--- BANTA BRANCH.prj (project) ---

Proj Title=BANTA BRANCH Base Level Engineering
Current Plan=p01
Default Exp/Contr=0.3,0.1
English Units
Geom File=g01
Flow File=f01
Plan File=p01
BEGIN DESCRIPTION:
BANTA BRANCH
END DESCRIPTION:

--- BANTA BRANCH.p01 (plan) ---

Plan Title=Multiple Run
Short Identifier=Multiple
Geom File=g01
Flow File=f01
Subcritical Flow
K Sum by GR= 0
Std Step Tol= 0.01
Critical Tol= 0.01
Num of Std Step Trials= 20
Max Error Tol= 0.3
Flow Tol Ratio= 0.001
Split Flow NTrial= 30
Split Flow Tol= 0.02
Split Flow Ratio= 0.02
Log Output Level= 0
Friction Slope Method= 1
Unsteady Friction Slope Method= 2
Unsteady Bridges Friction Slope Method= 1
Parabolic Critical Depth
Global Vel Dist=  1 , 1 , 1
Global Log Level= 0
CheckData=True
Encroach Param= -1, 0, 0, 0
BEGIN DESCRIPTION:
Multiple Run
END DESCRIPTION:

--- BANTA BRANCH.f01 (steady flow) ---

Flow Title=Multiple
Number of Profiles=7
Profile Names=10-year,25-year,50-year,1pct_min,100-year,1pct_plu,500-year
River Rch & RM= BANTA BRANCH,Reach-1,19918
    1819    2705    3483    3261    4410    5964    7078
River Rch & RM= BANTA BRANCH,Reach-1,14760
    2155    3225    4171    3918    5299    7167    8566
River Rch & RM= BANTA BRANCH,Reach-1,10533
    2675    4037    5250    4956    6703    9065   10942
River Rch & RM= BANTA BRANCH,Reach-1,7447
    2783    4213    5491    5195    7026    9502   11519
River Rch & RM= BANTA BRANCH,Reach-1,5542
    2972    4509    5884    5574    7538   10194   12387
River Rch & RM= BANTA BRANCH,Reach-1,518
    3404    5195    6808    6472    8753   11838   14492
Boundary for River Rch & Prof#=BANTA BRANCH,Reach-1,1
Up Type=0
Dn Type=3
Dn Slope=0.005
Boundary for River Rch & Prof#=BANTA BRANCH,Reach-1,2
Up Type=0
Dn Type=3
Dn Slope=0.005
Boundary for River Rch & Prof#=BANTA BRANCH,Reach-1,3
Up Type=0
Dn Type=3
Dn Slope=0.005
Boundary for River Rch & Prof#=BANTA BRANCH,Reach-1,4
Up Type=0
Dn Type=3
Dn Slope=0.005
Boundary for River Rch & Prof#=BANTA BRANCH,Reach-1,5
Up Type=0
Dn Type=3
Dn Slope=0.005
Boundary for River Rch & Prof#=BANTA BRANCH,Reach-1,6
Up Type=0
Dn Type=3
Dn Slope=0.005
Boundary for River Rch & Prof#=BANTA BRANCH,Reach-1,7
Up Type=0
Dn Type=3
Dn Slope=0.005

--- BANTA BRANCH.g01 (geometry) ---

Geom Title=Existing Conditions

River Reach=BANTA BRANCH,Reach-1
Reach XY= 30
      2645908.47     10085013.73      2645972.56     10084319.91
      2645790.09     10084119.00      2646190.87     10083340.41
      2646063.43     10083163.34      2645979.22     10082208.90
      2646055.49     10081544.90      2645772.16     10081172.14
      2645730.43     10080666.14      2645078.47     10080053.73
      2644918.47     10079023.73      2643990.32     10078322.97
      2643804.85     10077595.29      2643469.90     10077118.13
      2643456.80     10076741.60      2643136.44     10075826.96
      2642660.05     10075556.10      2642731.28     10075040.88
      2642454.12     10074513.27      2642475.74     10074152.66
      2642772.35     10073415.27      2643675.85     10072532.65
      2644054.73     10071553.23      2644351.32     10071379.18
      2644615.31     10070851.36      2645345.84     10070248.77
      2645825.10     10070025.63      2646113.50     10069696.22
      2646391.53     10069083.34      2646288.47     10068723.73

Type RM Length L Ch R = 1,19918,412,412,412
BEGIN DESCRIPTION:
BANTA BRANCH 44.0
END DESCRIPTION:
XS GIS Cut Line= 2
      2646281.50     10084957.15      2645471.73     10084893.07
#Sta/Elev= 30
  4632.5 2121.92  4705.8 2119.79  4724.2 2119.44  4735.0 2118.76  4740.1 2118.95
  4765.9 2115.22  4776.0 2114.16  4796.0 2113.00  4868.6 2111.25  4886.3 2111.25
  4926.4 2109.97  4956.5 2108.26  4976.6 2108.12  4986.6 2108.48  4994.2 2107.73
  4997.0 2107.23  5000.2 2107.73  5016.7 2108.88  5056.9 2109.34  5086.9 2109.01
  5115.8 2109.77  5120.8 2109.56  5147.1 2110.53  5237.4 2112.56  5277.5 2116.15
  5327.7 2119.17  5357.8 2120.64  5387.9 2121.57  5418.0 2124.25  5444.8 2126.07
#Mann=5,-1,0
  4632.5     0.1       0  4705.8    0.16       0  4724.2     0.1       0
  4994.2    0.07       0  5000.2     0.1       0
Bank Sta=4994.2,5000.2
Exp/Cntr=0.3,0.1

Type RM Length L Ch R = 1,19506,455,455,455
BEGIN DESCRIPTION:
BANTA BRANCH 43.0
END DESCRIPTION:
XS GIS Cut Line= 2
      2646332.85     10084585.22      2645447.45     10084449.81
#Sta/Elev= 30
  4638.3 2119.53  4794.5 2116.79  4857.9 2113.53  4864.0 2113.25  4885.5 2111.30
  4943.5 2107.47  4966.5 2106.34  4976.6 2106.40  4986.7 2105.57  4993.8 2104.13
  4996.6 2103.63  4999.8 2104.13  5006.9 2104.86  5012.0 2104.72  5017.0 2105.63
  5027.2 2105.94  5087.9 2106.26  5148.9 2105.71  5168.8 2106.42  5207.3 2109.17
  5212.3 2108.95  5249.7 2111.37  5275.8 2113.74  5290.2 2114.38  5320.5 2117.40
  5412.7 2121.08  5476.1 2124.58  5482.4 2125.59  5502.6 2127.08  5534.0 2128.36
#Mann=5,-1,0
  4638.3     0.1       0  4857.9    0.16       0  4864.0     0.1       0
  4993.8    0.07       0  4999.8     0.1       0
Bank Sta=4993.8,4999.8
Exp/Cntr=0.3,0.1

Type RM Length L Ch R = 1,19051,52,52,52
BEGIN DESCRIPTION:
Mapping XS 2b5c7267
END DESCRIPTION:
XS GIS Cut Line= 2
      2646553.37     10084203.28      2645501.55     10084151.30
#Sta/Elev= 30
  4257.1 2118.95  4292.0 2117.80  4392.2 2115.75  4442.2 2113.94  4512.3 2113.51
  4593.2 2110.17  4632.5 2108.16  4663.1 2107.04  4712.6 2105.64  4852.7 2103.87
  4862.7 2103.27  4892.8 2100.36  4912.8 2096.49  4949.4 2095.30  4952.2 2094.80
  4955.4 2095.30  4957.4 2095.73  4982.9 2095.94  5012.9 2097.29  5022.9 2098.01
  5032.9 2100.89  5043.0 2106.38  5053.0 2109.65  5103.0 2115.70  5123.1 2117.41
  5173.1 2119.10  5203.2 2120.95  5219.2 2122.36  5243.2 2124.29  5310.2 2127.45
#Mann=6,-1,0
  4257.1     0.1       0  4593.2    0.16       0  4663.1     0.1       0
  4949.4    0.07       0  4955.4     0.1       0  5219.2    0.16       0
Bank Sta=4949.4,4955.4
Exp/Cntr=0.3,0.1

Type RM Length L Ch R = 1,18999,45,45,45
BEGIN DESCRIPTION:
BANTA BRANCH 42.0
END DESCRIPTION:
XS GIS Cut Line= 2
      2646586.40     10084156.41      2645506.52     10084109.53
#Sta/Elev= 30
  4202.9 2120.87  4290.9 2116.68  4351.0 2115.67  4461.1 2111.86  4533.0 2110.39
  4563.9 2109.41  4641.2 2106.62  4781.4 2104.11  4851.4 2103.42  4861.5 2104.60
  4871.5 2107.31  4881.5 2108.29  4921.5 2105.88  4941.5 2106.17  4951.5 2105.37
  4961.5 2103.40  4981.6 2101.36  4998.6 2097.37  5001.3 2096.87  5004.6 2097.37
  5021.6 2104.48  5061.6 2110.73  5069.2 2113.01  5074.2 2112.58  5081.7 2114.45
  5091.7 2115.92  5141.7 2118.37  5217.2 2124.05  5241.8 2125.57  5283.8 2127.04
#Mann=6,-1,0
  4202.9     0.1       0  4533.0    0.16       0  4563.9     0.1       0
  4998.6    0.07       0  5004.6     0.1       0  5217.2    0.16       0
Bank Sta=4998.6,5004.6
Exp/Cntr=0.3,0.1

Type RM Length L Ch R = 1,18954,460,460,460
BEGIN DESCRIPTION:
Mapping XS 3c1d4908
END DESCRIPTION:
XS GIS Cut Line= 2
      2646555.07     10084113.00      2645527.33     10084066.13
#Sta/Elev= 30
  4249.1 2118.55  4255.7 2118.01  4315.8 2115.74  4335.8 2115.43  4365.8 2114.43
  4475.9 2112.30  4492.7 2111.50  4546.0 2109.61  4576.9 2108.95  4666.1 2106.29
  4766.2 2104.50  4781.5 2103.92  4816.3 2103.33  4916.4 2102.75  4956.4 2102.17
  4976.5 2101.18  4986.5 2100.05  4998.4 2098.22  5001.1 2097.72  5004.4 2098.22
  5016.5 2101.87  5026.5 2106.21  5036.5 2109.37  5046.5 2111.20  5076.6 2115.07
  5146.6 2118.42  5221.2 2123.50  5226.7 2124.20  5252.2 2125.31  5277.9 2126.35
#Mann=6,-1,0
  4249.1     0.1       0  4492.7    0.16       0  4576.9     0.1       0
  4998.4    0.07       0  5004.4     0.1       0  5252.2    0.16       0
Bank Sta=4998.4,5004.4
Exp/Cntr=0.3,0.1

Type RM Length L Ch R = 1,18494,422,422,422
BEGIN DESCRIPTION:
BANTA BRANCH 41.0
END DESCRIPTION:
XS GIS Cut Line= 3
      2646418.45     10083903.72      2646018.47     10083703.73
      2645818.46     10083703.73
#Sta/Elev= 30
  4541.7 2112.65  4578.0 2111.14  4639.5 2107.17  4661.9 2106.32  4689.8 2104.44
  4712.2 2103.80  4741.1 2103.45  4801.6 2102.07  4854.7 2101.25  4863.1 2100.84
  4899.5 2100.78  4935.8 2099.91  4980.5 2098.12  4986.1 2097.29  4991.4 2097.29
  4995.9 2095.13  4998.6 2094.63  5001.9 2095.13  5008.9 2095.61  5018.9 2097.60
  5048.9 2098.42  5078.9 2098.59  5088.9 2099.21  5108.9 2104.84  5118.9 2106.52
  5138.9 2109.01  5158.9 2110.81  5168.9 2112.04  5178.9 2112.88  5188.9 2113.16
#Mann=4,-1,0
  4541.7    0.16       0  4741.1     0.1       0  4995.9    0.07       0
  5001.9     0.1       0
Bank Sta=4995.9,5001.9
Exp/Cntr=0.3,0.1

Type RM Length L Ch R = 1,18072,514,514,514
BEGIN DESCRIPTION:
BANTA BRANCH 40.0
END DESCRIPTION:
XS GIS Cut Line= 4
      2646699.21     10083449.81      2646374.56     10083310.92
      2645900.60     10083354.32      2645667.97     10083397.73
#Sta/Elev= 30
  4462.2 2111.22  4574.1 2107.58  4613.7 2106.19  4666.3 2103.60  4785.6 2099.19
  4851.6 2097.54  4962.0 2096.01  4972.1 2094.31  4989.1 2088.58  4991.9 2088.08
  4995.1 2088.58  5002.2 2089.10  5008.9 2091.66  5013.9 2090.61  5022.3 2092.94
  5032.3 2094.21  5052.4 2093.96  5072.5 2094.58  5102.6 2094.65  5119.0 2095.67
  5162.9 2097.25  5182.9 2098.89  5213.1 2102.56  5229.0 2103.80  5273.3 2105.25
  5354.5 2106.79  5369.8 2108.14  5385.0 2108.48  5422.5 2111.52  5527.9 2113.73
#Mann=5,-1,0
  4462.2     0.1       0  4574.1    0.16       0  4785.6     0.1       0
  4989.1    0.07       0  4995.1     0.1       0
Bank Sta=4989.1,4995.1
Exp/Cntr=0.3,0.1

Type RM Length L Ch R = 1,17558,371,371,371
BEGIN DESCRIPTION:
BANTA BRANCH 39.0
END DESCRIPTION:
XS GIS Cut Line= 2
      2646579.45     10082868.21      2645683.58     10082875.16
#Sta/Elev= 30
  4519.2 2107.81  4540.2 2107.24  4560.2 2106.23  4580.2 2105.59  4620.2 2103.62
  4720.2 2100.14  4733.2 2099.27  4750.2 2097.99  4770.2 2095.93  4800.2 2094.60
  4910.2 2092.34  4970.2 2091.37  4980.2 2088.44  4997.2 2085.96  5000.0 2085.46
  5003.2 2085.96  5010.2 2086.79  5020.2 2088.95  5040.2 2091.25  5100.2 2092.95
  5120.2 2092.72  5130.2 2092.17  5140.2 2092.55  5170.2 2095.60  5220.2 2098.52
  5260.2 2100.35  5310.2 2103.65  5400.2 2108.88  5410.2 2110.00  5415.1 2110.00
#Mann=4,-1,0
  4519.2    0.16       0  4733.2     0.1       0  4997.2    0.07       0
  5003.2     0.1       0
Bank Sta=4997.2,5003.2
Exp/Cntr=0.3,0.1

Type RM Length L Ch R = 1,17187,464,464,464
BEGIN DESCRIPTION:
BANTA BRANCH 38.0
END DESCRIPTION:
XS GIS Cut Line= 2
      2646377.63     10082461.09      2645574.65     10082580.45
#Sta/Elev= 30
  4638.5 2097.80  4668.0 2095.87  4769.1 2092.30  4809.5 2091.47  4860.1 2091.06
  4880.3 2090.22  4895.0 2090.18  4959.3 2088.20  4971.3 2088.08  4981.4 2087.37
  4991.5 2084.72  4998.6 2082.20  5001.4 2081.70  5004.6 2082.20  5011.7 2083.96
  5021.8 2087.82  5028.7 2089.56  5042.0 2089.72  5098.1 2088.44  5112.8 2088.38
  5167.5 2088.83  5183.6 2089.33  5193.7 2090.06  5203.8 2091.38  5231.8 2095.89
  5236.9 2095.77  5274.6 2097.77  5294.8 2098.37  5375.7 2104.11  5450.3 2106.99
#Mann=3,-1,0
  4638.5     0.1       0  4998.6    0.07       0  5004.6     0.1       0
Bank Sta=4998.6,5004.6
Exp/Cntr=0.3,0.1

Type RM Length L Ch R = 1,16723,455,455,455
BEGIN DESCRIPTION:
BANTA BRANCH 37.0
END DESCRIPTION:
XS GIS Cut Line= 3
      2646418.43     10082103.73      2645968.47     10082053.73
      2645568.51     10082253.71
#Sta/Elev= 30
  4554.0 2098.20  4584.1 2097.54  4644.5 2093.93  4785.4 2089.92  4886.0 2087.65
  4906.1 2086.85  4936.3 2085.07  4966.5 2084.82  4986.6 2083.06  4993.7 2082.82
  4996.4 2082.32  4999.7 2082.82  5015.1 2083.29  5020.7 2082.97  5029.1 2084.09
  5043.1 2085.30  5065.4 2085.77  5149.3 2084.86  5163.3 2085.00  5261.1 2088.05
  5266.7 2088.79  5283.4 2088.56  5289.0 2089.45  5305.8 2089.42  5311.4 2089.90
  5333.8 2090.55  5417.6 2092.39  5431.6 2093.38  5451.1 2099.34  5453.9 2099.34
#Mann=3,-1,0
  4554.0     0.1       0  4993.7    0.07       0  4999.7     0.1       0
Bank Sta=4993.7,4999.7
Exp/Cntr=0.3,0.1

Type RM Length L Ch R = 1,16268,348,348,348
BEGIN DESCRIPTION:
BANTA BRANCH 36.0
END DESCRIPTION:
XS GIS Cut Line= 3
      2646488.73     10081688.80      2646129.33     10081610.67
      2645275.15     10081902.34
#Sta/Elev= 30
  4566.9 2099.24  4606.9 2098.53  4697.9 2095.23  4741.1 2093.06  4800.0 2087.35
  4823.0 2086.11  4884.4 2084.10  4960.8 2084.24  4983.9 2078.50  4986.6 2078.00
  4989.9 2078.50  4992.2 2079.60  4999.0 2078.56  5009.6 2079.05  5018.2 2081.35
  5023.5 2081.58  5054.8 2081.56  5104.7 2079.90  5180.1 2082.00  5231.5 2081.66
  5263.2 2082.32  5456.7 2087.54  5488.0 2090.10  5537.9 2091.70  5569.6 2093.85
  5608.1 2097.49  5728.1 2104.14  5764.7 2107.29  5802.1 2111.56  5837.3 2113.32
#Mann=5,-1,0
  4566.9     0.1       0  4606.9    0.16       0  4697.9     0.1       0
  4983.9    0.07       0  4989.9     0.1       0
Bank Sta=4983.9,4989.9
Exp/Cntr=0.3,0.1

Type RM Length L Ch R = 1,15920,575,575,575
BEGIN DESCRIPTION:
BANTA BRANCH 35.0
END DESCRIPTION:
XS GIS Cut Line= 3
      2646509.53     10081444.00      2645952.25     10081313.80
      2645238.71     10081694.00
#Sta/Elev= 30
  4358.7 2096.57  4378.0 2096.19  4503.6 2093.48  4544.9 2091.90  4575.4 2090.30
  4596.0 2088.03  4601.4 2086.86  4637.1 2084.30  4739.8 2081.71  4776.6 2081.86
  4936.0 2079.99  4957.5 2078.38  4969.3 2078.24  4998.4 2074.65  5001.2 2074.15
  5004.4 2074.65  5023.4 2077.54  5037.3 2078.42  5089.3 2077.49  5133.2 2078.80
  5161.9 2081.11  5177.1 2081.74  5399.8 2085.72  5467.6 2087.54  5517.2 2090.39
  5555.5 2093.21  5599.4 2097.33  5670.1 2101.88  5700.0 2104.45  5739.5 2108.70
#Mann=7,-1,0
  4358.7     0.1       0  4378.0    0.16       0  4544.9     0.1       0
  4998.4    0.07       0  5004.4     0.1       0  5670.1    0.16       0
  5700.0     0.1       0
Bank Sta=4998.4,5004.4
Exp/Cntr=0.3,0.1

Type RM Length L Ch R = 1,15345,585,585,585
BEGIN DESCRIPTION:
BANTA BRANCH 34.0
END DESCRIPTION:
XS GIS Cut Line= 3
      2646479.58     10081057.01      2645902.34     10080798.77
      2645196.76     10080989.23
#Sta/Elev= 30
  4272.2 2087.79  4291.2 2087.61  4372.0 2085.39  4459.0 2084.05  4510.9 2082.76
  4547.3 2082.66  4586.0 2081.69  4655.6 2080.97  4661.1 2080.62  4712.9 2080.11
  4788.3 2080.00  4828.9 2078.88  4943.8 2076.75  4970.7 2075.28  4978.5 2073.93
  4983.7 2073.98  4991.4 2071.42  4998.8 2070.21  5001.6 2069.71  5004.8 2070.21
  5012.2 2071.37  5018.4 2072.83  5058.3 2073.94  5084.7 2074.08  5105.4 2075.07
  5281.5 2075.51  5362.0 2076.43  5467.9 2078.63  5530.1 2080.59  5635.4 2084.57
#Mann=3,-1,0
  4272.2     0.1       0  4998.8    0.07       0  5004.8     0.1       0
Bank Sta=4998.8,5004.8
Exp/Cntr=0.3,0.1

Type RM Length L Ch R = 1,14760,301,301,301
BEGIN DESCRIPTION:
BANTA BRANCH 33.0
END DESCRIPTION:
XS GIS Cut Line= 3
      2645962.64     10080194.01      2645493.91     10080350.26
      2645035.58     10080824.21
#Sta/Elev= 30
  4402.5 2087.60  4572.9 2082.05  4604.5 2081.21  4641.4 2080.71  4699.4 2078.23
  4762.6 2074.26  4775.8 2074.05  4839.1 2071.76  4870.7 2071.29  4881.2 2071.42
  4910.0 2070.85  4945.2 2069.00  4973.5 2068.65  4980.7 2068.37  4998.8 2065.77
  5001.6 2065.27  5004.8 2065.77  5009.0 2068.60  5016.0 2070.43  5023.2 2070.92
  5058.4 2070.32  5086.7 2070.62  5185.8 2073.13  5207.1 2074.05  5214.1 2074.62
  5235.3 2075.23  5263.5 2077.53  5327.2 2079.26  5440.4 2084.21  5555.9 2088.05
#Mann=3,-1,0
  4402.5     0.1       0  4998.8    0.07       0  5004.8     0.1       0
Bank Sta=4998.8,5004.8
Exp/Cntr=0.3,0.1

Type RM Length L Ch R = 1,14459,439,439,439
BEGIN DESCRIPTION:
BANTA BRANCH 32.0
END DESCRIPTION:
XS GIS Cut Line= 3
      2645618.45     10079953.74      2645218.47     10080203.73
      2644968.50     10080403.71
#Sta/Elev= 30
  4532.6 2078.88  4555.6 2077.50  4619.3 2074.82  4634.6 2073.26  4671.1 2071.33
  4802.0 2069.85  4815.6 2070.12  4954.2 2069.41  4968.9 2068.49  4981.3 2065.54
  4990.7 2064.18  4993.6 2063.36  4996.4 2062.86  4999.6 2063.36  5001.3 2063.81
  5007.5 2063.81  5017.9 2065.46  5040.3 2067.18  5061.1 2067.62  5096.3 2067.15
  5160.4 2072.46  5174.8 2073.28  5203.6 2074.08  5210.0 2075.00  5218.0 2075.14
  5224.4 2075.85  5232.4 2075.87  5238.8 2076.61  5274.0 2077.89  5324.4 2078.82
#Mann=3,-1,0
  4532.6     0.1       0  4993.6    0.07       0  4999.6     0.1       0
Bank Sta=4993.6,4999.6
Exp/Cntr=0.3,0.1

Type RM Length L Ch R = 1,14020,461,461,461
BEGIN DESCRIPTION:
BANTA BRANCH 31.0
END DESCRIPTION:
XS GIS Cut Line= 3
      2645514.76     10079563.79      2644926.21     10079891.92
      2644738.73     10080115.86
#Sta/Elev= 30
  4428.7 2077.97  4543.1 2076.02  4564.8 2074.66  4586.5 2072.07  4653.4 2067.25
  4683.7 2066.57  4764.8 2066.41  4814.0 2066.81  4846.0 2065.66  4905.3 2064.85
  4911.1 2063.60  4916.8 2063.52  4927.1 2062.39  4962.6 2063.11  4970.5 2062.94
  4992.3 2061.22  5011.0 2060.91  5013.7 2060.41  5017.0 2060.91  5019.8 2062.53
  5030.0 2065.02  5042.7 2066.93  5057.4 2067.82  5095.1 2069.15  5137.7 2069.94
  5201.5 2073.34  5215.8 2073.64  5279.6 2076.62  5357.6 2078.37  5394.6 2078.70
#Mann=3,-1,0
  4428.7     0.1       0  5011.0    0.07       0  5017.0     0.1       0
Bank Sta=5011,5017
Exp/Cntr=0.3,0.1

Type RM Length L Ch R = 1,13559,451,451,451
BEGIN DESCRIPTION:
BANTA BRANCH 30.0
END DESCRIPTION:
XS GIS Cut Line= 3
      2645405.39     10079329.42      2644915.79     10079428.38
      2644566.82     10079735.69
#Sta/Elev= 30
  4605.0 2076.67  4631.1 2076.06  4683.5 2075.22  4734.5 2072.67  4785.5 2068.09
  4802.1 2066.07  4867.1 2062.14  4908.7 2061.87  4979.3 2063.59  4989.6 2059.28
  4996.8 2057.90  4999.5 2057.40  5002.8 2057.90  5010.2 2058.52  5020.2 2060.59
  5040.6 2061.63  5081.4 2059.89  5091.6 2058.40  5104.5 2058.84  5113.9 2061.84
  5127.6 2063.26  5235.3 2064.48  5261.9 2064.52  5340.6 2066.16  5375.7 2068.11
  5418.4 2071.93  5443.1 2073.45  5488.7 2075.28  5517.1 2075.67  5569.5 2077.47
#Mann=6,-1,0
  4605.0    0.16       0  4631.1     0.1       0  4996.8    0.07       0
  5002.8     0.1       0  5235.3    0.16       0  5443.1     0.1       0
Bank Sta=4996.8,5002.8
Exp/Cntr=0.3,0.1

Type RM Length L Ch R = 1,13108,439,439,439
BEGIN DESCRIPTION:
BANTA BRANCH 29.0
END DESCRIPTION:
XS GIS Cut Line= 3
      2645405.35     10078970.04      2644947.04     10078917.96
      2644427.17     10079489.82
#Sta/Elev= 30
  4449.4 2075.17  4481.7 2074.58  4526.8 2073.30  4545.7 2073.25  4550.8 2072.87
  4640.3 2071.27  4724.9 2067.89  4788.5 2066.94  4907.4 2064.13  4949.0 2063.94
  4963.2 2062.79  4977.4 2061.08  4996.0 2053.98  4998.7 2053.48  5002.0 2053.98
  5013.1 2055.75  5026.7 2056.34  5048.3 2058.68  5076.7 2059.55  5168.6 2060.58
  5380.8 2061.05  5430.8 2062.01  5465.9 2064.27  5551.0 2068.81  5572.0 2069.53
  5614.6 2072.20  5621.3 2072.25  5628.8 2073.15  5635.5 2073.18  5683.5 2075.61
#Mann=4,-1,0
  4449.4    0.16       0  4481.7     0.1       0  4996.0    0.07       0
  5002.0     0.1       0
Bank Sta=4996,5002
Exp/Cntr=0.3,0.1

Type RM Length L Ch R = 1,12669,441,441,441
BEGIN DESCRIPTION:
BANTA BRANCH 28.0
END DESCRIPTION:
XS GIS Cut Line= 3
      2644918.46     10078353.74      2644518.47     10078753.73
      2644168.45     10079153.75
#Sta/Elev= 30
  4435.5 2067.45  4562.8 2063.73  4702.6 2060.65  4774.9 2059.44  4845.6 2059.40
  4888.0 2057.92  4902.2 2056.74  4916.3 2058.51  4930.5 2059.25  4958.7 2057.74
  4987.0 2053.23  4994.6 2052.40  4997.4 2051.90  5000.6 2052.40  5004.5 2052.40
  5008.3 2053.70  5022.5 2055.42  5071.9 2055.98  5093.7 2056.86  5135.5 2056.78
  5185.8 2058.28  5256.0 2057.73  5313.0 2058.24  5333.8 2059.03  5348.1 2060.37
  5355.7 2061.78  5369.9 2063.47  5419.3 2066.57  5525.6 2070.85  5532.7 2071.24
#Mann=5,-1,0
  4435.5    0.16       0  4702.6     0.1       0  4994.6    0.07       0
  5000.6     0.1       0  5525.6    0.16       0
Bank Sta=4994.6,5000.6
Exp/Cntr=0.3,0.1

Type RM Length L Ch R = 1,12228,428,428,428
BEGIN DESCRIPTION:
BANTA BRANCH 27.0
END DESCRIPTION:
XS GIS Cut Line= 3
      2644968.46     10078203.73      2644168.47     10078503.73
      2643818.47     10078903.73
#Sta/Elev= 30
  4125.9 2071.46  4196.2 2069.02  4281.6 2067.26  4318.1 2065.53  4526.6 2061.88
  4591.0 2060.66  4648.3 2059.55  4659.9 2058.78  4708.8 2057.69  4764.0 2055.77
  4894.9 2054.06  4916.2 2052.98  4983.6 2052.13  4994.1 2051.35  5015.9 2052.10
  5033.8 2051.06  5036.5 2050.56  5039.8 2051.06  5044.4 2051.88  5051.0 2053.92
  5058.6 2054.78  5072.8 2055.48  5108.0 2056.35  5257.0 2057.85  5285.4 2058.58
  5292.1 2058.93  5320.6 2062.31  5334.8 2063.30  5369.9 2064.45  5511.8 2071.46
#Mann=5,-1,0
  4125.9     0.1       0  4526.6    0.16       0  4591.0     0.1       0
  5033.8    0.07       0  5039.8     0.1       0
Bank Sta=5033.8,5039.8
Exp/Cntr=0.3,0.1

Type RM Length L Ch R = 1,11800,377,377,377
BEGIN DESCRIPTION:
BANTA BRANCH 26.0
END DESCRIPTION:
XS GIS Cut Line= 3
      2644551.17     10077938.81      2643832.46     10078214.84
      2643530.36     10078704.44
#Sta/Elev= 30
  4327.3 2065.39  4355.6 2064.85  4463.1 2062.69  4465.2 2062.66  4520.0 2060.79
  4598.0 2059.32  4659.9 2057.36  4774.1 2054.50  4823.0 2052.81  4846.1 2051.33
  4865.8 2050.07  4919.4 2050.99  4973.4 2049.26  4983.6 2048.22  4995.1 2045.95
  4997.8 2045.45  5001.1 2045.95  5015.8 2049.00  5022.8 2050.86  5028.1 2051.51
  5058.6 2052.65  5099.5 2052.54  5223.9 2054.02  5272.3 2053.89  5324.4 2054.78
  5376.5 2056.55  5403.6 2058.63  5541.9 2062.71  5571.6 2063.59  5672.5 2068.98
#Mann=9,-1,0
  4327.3     0.1       0  4355.6    0.16       0  4463.1     0.1       0
  4465.2    0.16       0  4659.9     0.1       0  4846.1    0.05       0
  4995.1   0.035       0  5001.1    0.05       0  5541.9     0.1       0
Bank Sta=4995.1,5001.1
Exp/Cntr=0.3,0.1

Type RM Length L Ch R = 1,11423,380,380,380
BEGIN DESCRIPTION:
BANTA BRANCH 25.0
END DESCRIPTION:
XS GIS Cut Line= 3
      2644580.70     10077608.67      2643899.30     10077775.77
      2643452.24     10078220.66
#Sta/Elev= 30
  4213.6 2065.27  4288.0 2064.40  4308.6 2063.47  4425.4 2061.28  4503.4 2059.27
  4566.0 2058.75  4751.3 2054.76  4792.5 2053.49  4804.8 2052.69  4823.4 2050.25
  4841.3 2046.19  4846.4 2045.81  4879.6 2047.13  4893.2 2047.15  4963.8 2047.89
  4978.0 2046.87  4985.1 2045.56  5003.3 2044.50  5006.0 2044.00  5009.3 2044.50
  5013.4 2045.78  5027.5 2048.33  5034.5 2048.85  5125.7 2050.18  5161.8 2051.83
  5183.1 2052.04  5190.1 2051.55  5246.7 2051.31  5430.5 2052.39  5545.9 2054.60
#Mann=6,-1,0
  4213.6     0.1       0  4879.6    0.05       0  4893.2     0.1       0
  5003.3    0.07       0  5009.3     0.1       0  5125.7    0.05       0
Bank Sta=5003.3,5009.3
Exp/Cntr=0.3,0.1

Type RM Length L Ch R = 1,11043,510,510,510
BEGIN DESCRIPTION:
BANTA BRANCH 24.0
END DESCRIPTION:
XS GIS Cut Line= 3
      2644223.03     10077308.61      2643587.66     10077548.17
      2643165.78     10078615.91
#Sta/Elev= 30
  4476.7 2059.05  4716.7 2054.06  4770.1 2050.88  4842.6 2049.22  4872.8 2046.20
  4887.7 2045.77  4941.1 2046.58  4963.4 2046.15  5002.3 2042.16  5005.0 2041.66
  5008.3 2042.16  5026.6 2044.16  5068.2 2044.40  5103.7 2048.03  5155.7 2047.68
  5251.0 2049.20  5473.5 2049.75  5516.0 2050.84  5545.8 2052.50  5551.2 2053.60
  5581.1 2054.88  5654.0 2054.70  5737.8 2056.16  5846.0 2056.70  5905.4 2058.81
  6000.4 2060.47  6054.8 2062.71  6181.4 2069.42  6224.6 2071.26  6303.8 2072.73
#Mann=5,-1,0
  4476.7     0.1       0  5002.3    0.07       0  5008.3     0.1       0
  6054.8    0.05       0  6181.4     0.1       0
Bank Sta=5002.3,5008.3
Exp/Cntr=0.3,0.1

Type RM Length L Ch R = 1,10533,545,545,545
BEGIN DESCRIPTION:
BANTA BRANCH 23.0
END DESCRIPTION:
XS GIS Cut Line= 3
      2644203.66     10076926.63      2643634.83     10077072.25
      2642263.40     10077164.52
#Sta/Elev= 30
  4237.9 2061.36  4609.5 2051.88  4718.1 2045.96  4726.8 2044.85  4759.4 2044.24
  4820.6 2041.61  4911.6 2042.88  4971.8 2042.02  4986.1 2040.07  4998.8 2038.39
  5001.6 2037.89  5004.8 2038.39  5021.9 2039.39  5041.9 2043.26  5051.9 2043.73
  5102.1 2045.04  5177.5 2044.84  5379.6 2045.91  5478.8 2047.10  5517.8 2048.57
  5543.1 2051.02  5553.1 2050.93  5633.3 2054.82  5693.4 2058.43  5783.6 2061.31
  5863.8 2062.85  5893.8 2064.29  5933.9 2067.68  5974.0 2069.39  6199.6 2075.76
#Mann=7,-1,0
  4237.9     0.1       0  4986.1    0.16       0  4998.8    0.07       0
  5004.8    0.16       0  5177.5     0.1       0  5379.6    0.05       0
  5478.8     0.1       0
Bank Sta=4998.8,5004.8
Exp/Cntr=0.3,0.1

Type RM Length L Ch R = 1,9988,383,383,383
BEGIN DESCRIPTION:
BANTA BRANCH 22.0
END DESCRIPTION:
XS GIS Cut Line= 3
      2643952.29     10076579.43      2643457.46     10076542.96
      2642535.59     10076850.25
#Sta/Elev= 30
  4438.7 2056.94  4595.3 2052.10  4693.9 2048.73  4713.3 2047.12  4792.5 2045.49
  4891.1 2041.50  4944.3 2039.27  4966.2 2036.36  4994.1 2033.10  4996.8 2032.60
  5000.1 2033.10  5007.6 2033.83  5014.6 2036.67  5046.2 2037.77  5102.5 2036.00
  5146.4 2038.80  5186.8 2039.98  5310.4 2040.82  5415.9 2042.00  5521.5 2043.98
  5557.5 2045.05  5576.8 2046.54  5589.1 2046.08  5640.0 2047.91  5678.7 2051.79
  5684.0 2051.47  5715.6 2053.69  5741.9 2056.92  5773.6 2058.62  5906.6 2062.65
#Mann=11,-1,0
  4438.7     0.1       0  4595.3    0.16       0  4693.9    0.05       0
  4792.5     0.1       0  4891.1    0.05       0  4966.2     0.1       0
  4994.1    0.07       0  5000.1     0.1       0  5310.4    0.16       0
  5415.9    0.05       0  5521.5     0.1       0
Bank Sta=4994.1,5000.1
Exp/Cntr=0.3,0.1

Type RM Length L Ch R = 1,9605,459,459,459
BEGIN DESCRIPTION:
BANTA BRANCH 21.0
END DESCRIPTION:
XS GIS Cut Line= 3
      2643837.71     10076048.16      2643176.21     10076230.46
      2642483.52     10076652.32
#Sta/Elev= 30
  4416.6 2054.70  4524.8 2051.75  4581.8 2049.94  4602.1 2047.47  4623.3 2046.94
  4664.8 2043.85  4686.5 2043.54  4778.9 2037.85  4862.1 2036.52  4903.1 2035.74
  4925.7 2033.25  4955.2 2033.79  4993.7 2031.20  4996.4 2030.70  4999.7 2031.20
  5027.8 2034.40  5056.2 2036.18  5124.0 2034.62  5213.1 2037.67  5339.0 2038.70
  5356.3 2039.00  5466.8 2041.14  5524.9 2043.12  5561.7 2045.58  5568.5 2044.23
  5591.9 2043.74  5641.2 2050.74  5693.4 2054.07  5825.1 2058.69  5913.8 2060.65
#Mann=8,-1,0
  4416.6    0.16       0  4524.8     0.1       0  4862.1    0.05       0
  4925.7     0.1       0  4993.7    0.07       0  4999.7     0.1       0
  5339.0    0.16       0  5356.3     0.1       0
Bank Sta=4993.7,4999.7
Exp/Cntr=0.3,0.1

Type RM Length L Ch R = 1,9146,375,375,375
BEGIN DESCRIPTION:
BANTA BRANCH 20.0
END DESCRIPTION:
XS GIS Cut Line= 4
      2643874.16     10075626.29      2643165.79     10075740.88
      2642467.87     10076246.09      2642463.03     10076246.09
#Sta/Elev= 30
  4208.1 2057.65  4355.7 2051.68  4453.3 2049.51  4538.7 2047.33  4671.4 2042.73
  4735.8 2041.26  4811.5 2039.05  4841.9 2038.99  4872.3 2037.42  4910.0 2034.58
  4915.1 2032.32  4975.5 2027.34  4990.2 2025.79  4993.4 2024.53  4996.2 2024.03
  4999.4 2024.53  5019.6 2025.79  5040.5 2030.09  5061.4 2031.56  5082.9 2032.13
  5105.5 2031.21  5155.8 2032.26  5226.9 2036.35  5255.7 2037.12  5448.9 2039.16
  5484.4 2041.23  5490.6 2042.27  5591.1 2044.51  5706.4 2050.34  5792.1 2053.26
#Mann=7,-1,0
  4208.1     0.1       0  4453.3    0.16       0  4538.7     0.1       0
  4671.4    0.16       0  4735.8     0.1       0  4993.4    0.07       0
  4999.4     0.1       0
Bank Sta=4993.4,4999.4
Exp/Cntr=0.3,0.1

Type RM Length L Ch R = 1,8771,555,555,555
BEGIN DESCRIPTION:
BANTA BRANCH 19.0
END DESCRIPTION:
XS GIS Cut Line= 3
      2643874.17     10075334.62      2642921.00     10075532.55
      2642281.43     10076109.72
#Sta/Elev= 30
  3835.0 2057.98  3869.1 2056.42  3912.3 2055.39  3922.5 2054.37  3960.4 2053.82
  4201.5 2047.40  4310.6 2043.33  4688.7 2036.67  4752.9 2035.30  4860.8 2030.55
  4946.0 2029.53  4960.1 2027.89  4992.3 2022.02  4995.1 2021.52  4998.3 2022.02
  5023.7 2023.32  5030.4 2025.18  5037.9 2025.81  5080.5 2024.24  5094.7 2026.34
  5108.3 2031.07  5115.6 2034.58  5125.8 2037.01  5129.8 2037.96  5144.0 2038.84
  5226.4 2042.65  5299.5 2044.11  5335.3 2045.62  5639.5 2051.55  5670.0 2052.83
#Mann=9,-1,0
  3835.0     0.1       0  3869.1    0.16       0  3960.4     0.1       0
  4688.7    0.16       0  4752.9     0.1       0  4992.3    0.07       0
  4998.3     0.1       0  5125.8    0.05       0  5226.4     0.1       0
Bank Sta=4992.3,4998.3
Exp/Cntr=0.3,0.1

Type RM Length L Ch R = 1,8216,378,378,378
BEGIN DESCRIPTION:
BANTA BRANCH 18.0
END DESCRIPTION:
XS GIS Cut Line= 2
      2643208.84     10075168.75      2642174.13     10075182.64
#Sta/Elev= 30
  4516.2 2039.04  4586.6 2037.72  4636.6 2036.05  4736.6 2034.45  4766.6 2034.36
  4856.6 2032.87  4876.6 2032.19  4906.6 2029.83  4916.6 2028.47  4926.6 2026.94
  4936.6 2024.18  4946.6 2022.43  4966.6 2021.56  4976.6 2020.71  4986.6 2015.73
  4993.6 2015.30  4996.4 2014.80  4999.6 2015.30  5006.6 2015.81  5026.6 2018.87
  5036.6 2021.52  5046.6 2023.61  5076.6 2027.11  5156.6 2031.55  5246.6 2034.45
  5260.7 2035.20  5286.6 2037.54  5396.7 2040.26  5468.9 2042.58  5551.0 2044.79
#Mann=4,-1,0
  4516.2     0.1       0  4993.6    0.07       0  4999.6     0.1       0
  5468.9    0.16       0
Bank Sta=4993.6,4999.6
Exp/Cntr=0.3,0.1

Type RM Length L Ch R = 1,7838,278,278,278
BEGIN DESCRIPTION:
BANTA BRANCH 17.0
END DESCRIPTION:
XS GIS Cut Line= 2
      2642836.26     10074736.22      2642294.54     10074965.41
#Sta/Elev= 30
  4765.7 2030.23  4811.7 2030.13  4876.1 2030.33  4928.9 2029.44  4952.6 2028.48
  4958.7 2026.77  4969.6 2022.78  4976.2 2018.15  4981.7 2016.08  4996.9 2012.89
  4999.7 2012.39  5002.9 2012.89  5029.1 2019.49  5034.8 2020.02  5052.7 2020.19
  5099.9 2022.56  5105.6 2024.04  5129.2 2027.49  5134.7 2027.51  5152.9 2029.30
  5158.4 2029.31  5182.1 2031.19  5187.5 2031.16  5205.7 2032.83  5211.2 2032.94
  5241.1 2035.77  5264.0 2036.04  5311.4 2037.77  5317.1 2038.36  5353.9 2039.13
#Mann=4,-1,0
  4765.7    0.05       0  4811.7     0.1       0  4996.9    0.07       0
  5002.9     0.1       0
Bank Sta=4996.9,5002.9
Exp/Cntr=0.3,0.1

Type RM Length L Ch R = 1,7560,113,113,113
BEGIN DESCRIPTION:
Mapping XS aa31c049
END DESCRIPTION:
XS GIS Cut Line= 2
      2642810.17     10074606.02      2642127.86     10074579.98
#Sta/Elev= 30
  4663.1 2028.92  4704.8 2028.75  4734.9 2028.05  4764.9 2027.97  4814.9 2027.05
  4844.9 2027.11  4852.1 2026.62  4857.1 2025.30  4864.9 2024.78  4895.0 2023.47
  4945.0 2022.49  4955.0 2020.88  4965.0 2016.80  4975.0 2013.17  4985.0 2012.06
  5002.0 2010.92  5004.8 2010.42  5008.0 2010.92  5015.1 2011.50  5045.1 2016.22
  5055.1 2019.66  5065.1 2023.56  5075.1 2025.98  5085.1 2026.93  5113.3 2028.41
  5125.1 2029.54  5165.2 2031.62  5189.6 2032.40  5275.2 2036.62  5345.9 2039.42
#Mann=4,-1,0
  4663.1    0.05       0  5002.0    0.04       0  5008.0    0.05       0
  5189.6    0.08       0
Bank Sta=5002,5008
Exp/Cntr=0.3,0.1

Type RM Length L Ch R = 1,7447,162,162,162
BEGIN DESCRIPTION:
Mapping XS 7af9047d
END DESCRIPTION:
XS GIS Cut Line= 2
      2642950.86     10074501.86      2642117.45     10074470.60
#Sta/Elev= 30
  4508.2 2031.70  4540.6 2030.11  4600.7 2028.33  4840.8 2026.45  4857.1 2025.55
  4862.1 2024.87  4870.8 2024.46  4890.9 2022.71  4900.9 2022.34  4930.9 2020.08
  4950.9 2017.68  4970.9 2013.61  4980.9 2012.17  4990.9 2011.06  5000.9 2010.74
  5007.9 2010.05  5010.7 2009.55  5013.9 2010.05  5031.0 2013.89  5041.0 2015.63
  5071.0 2028.43  5081.0 2031.11  5091.0 2032.24  5125.7 2034.59  5161.1 2035.72
  5184.5 2037.28  5201.1 2038.37  5231.1 2039.57  5261.1 2039.79  5342.2 2041.97
#Mann=4,-1,0
  4508.2    0.05       0  5007.9    0.04       0  5013.9    0.05       0
  5184.5    0.08       0
Bank Sta=5007.9,5013.9
Exp/Cntr=0.3,0.1

Type RM Length L Ch R = 1,7285,440,440,440
BEGIN DESCRIPTION:
BANTA BRANCH 16.0
END DESCRIPTION:
XS GIS Cut Line= 2
      2642950.82     10074361.23      2642075.84     10074293.52
#Sta/Elev= 30
  4511.0 2030.50  4523.4 2030.64  4545.9 2029.43  4553.5 2029.72  4599.6 2027.49
  4633.7 2026.13  4794.2 2025.27  4914.6 2020.14  4924.6 2022.79  4930.9 2025.19
  4935.9 2025.08  4944.7 2022.19  4954.7 2017.54  4964.7 2014.17  4991.8 2009.96
  4994.6 2009.46  4997.8 2009.96  5004.8 2010.00  5014.9 2011.18  5024.9 2011.25
  5034.9 2010.39  5045.0 2013.39  5055.0 2020.10  5060.9 2026.11  5075.0 2030.66
  5145.2 2034.95  5175.3 2037.42  5215.5 2039.51  5285.7 2041.08  5388.6 2045.05
#Mann=4,-1,0
  4511.0    0.05       0  4599.6     0.1       0  4991.8    0.07       0
  4997.8     0.1       0
Bank Sta=4991.8,4997.8
Exp/Cntr=0.3,0.1

Type RM Length L Ch R = 1,6845,279,279,279
BEGIN DESCRIPTION:
BANTA BRANCH 15.0
END DESCRIPTION:
XS GIS Cut Line= 2
      2643160.28     10074106.26      2642118.60     10073745.15
#Sta/Elev= 30
  4375.7 2033.19  4463.7 2031.32  4536.4 2031.10  4557.5 2029.65  4676.4 2026.66
  4769.8 2022.42  4826.8 2021.39  4852.6 2021.99  4875.1 2021.58  4889.1 2020.93
  4928.0 2014.62  4951.3 2012.56  4970.3 2008.21  4977.2 2007.43  4999.1 2007.31
  5001.8 2006.81  5005.1 2007.31  5013.6 2008.44  5033.8 2013.07  5039.5 2015.78
  5065.3 2022.77  5070.6 2023.22  5076.2 2025.36  5107.9 2029.37  5171.4 2036.17
  5203.2 2037.81  5257.5 2039.44  5314.4 2042.86  5425.4 2046.79  5478.2 2047.90
#Mann=3,-1,0
  4375.7     0.1       0  4999.1    0.07       0  5005.1     0.1       0
Bank Sta=4999.1,5005.1
Exp/Cntr=0.3,0.1

Type RM Length L Ch R = 1,6566,626,626,626
BEGIN DESCRIPTION:
BANTA BRANCH 14.0
END DESCRIPTION:
XS GIS Cut Line= 2
      2643645.16     10074189.75      2641952.94     10073235.16
#Sta/Elev= 30
  3908.9 2038.39  3975.9 2036.99  4461.6 2030.77  4579.7 2028.94  4703.9 2025.85
  4754.7 2025.52  4871.4 2021.42  4930.7 2016.17  4961.4 2012.23  4984.2 2004.64
  4992.8 2002.59  4995.6 2002.09  4998.8 2002.59  5018.8 2004.70  5033.2 2005.23
  5041.8 2006.92  5054.9 2009.97  5064.7 2013.20  5070.8 2016.28  5092.4 2021.39
  5108.4 2026.36  5122.1 2029.02  5210.9 2034.94  5254.2 2036.95  5297.5 2037.76
  5372.7 2041.87  5592.9 2048.98  5702.0 2051.71  5804.5 2052.57  5851.8 2053.80
#Mann=4,-1,0
  3908.9    0.05       0  4461.6     0.1       0  4992.8    0.07       0
  4998.8     0.1       0
Bank Sta=4992.8,4998.8
Exp/Cntr=0.3,0.1

Type RM Length L Ch R = 1,5940,398,398,398
BEGIN DESCRIPTION:
BANTA BRANCH 13.0
END DESCRIPTION:
XS GIS Cut Line= 2
      2644079.18     10073755.72      2642386.87     10072768.53
#Sta/Elev= 30
  3775.3 2039.34  4084.9 2034.89  4319.7 2030.41  4597.6 2022.63  4713.9 2017.66
  4763.8 2013.84  4779.5 2014.04  4785.3 2013.15  4801.0 2014.79  4822.5 2014.79
  4838.2 2016.12  4875.4 2013.97  4902.7 2010.17  4933.8 2007.72  4961.4 2003.10
  4988.7 2000.24  4991.5 1999.74  4994.7 2000.24  5004.4 2001.53  5014.4 2004.92
  5020.1 2009.20  5026.5 2012.44  5066.9 2020.54  5084.7 2023.27  5153.2 2028.45
  5246.4 2032.47  5356.7 2035.56  5378.2 2035.25  5474.1 2037.68  5734.5 2041.32
#Mann=5,-1,0
  3775.3     0.1       0  4988.7    0.07       0  4994.7     0.1       0
  5066.9    0.16       0  5153.2     0.1       0
Bank Sta=4988.7,4994.7
Exp/Cntr=0.3,0.1

Type RM Length L Ch R = 1,5542,497,497,497
BEGIN DESCRIPTION:
BANTA BRANCH 12.0
END DESCRIPTION:
XS GIS Cut Line= 2
      2643701.89     10073189.56      2642938.02     10072585.42
#Sta/Elev= 30
  4516.6 2024.23  4530.7 2023.82  4551.5 2022.36  4665.3 2018.31  4772.7 2016.06
  4843.2 2013.75  4872.1 2013.29  4892.9 2012.07  4921.8 2009.17  4936.2 2007.41
  4942.6 2005.80  4957.0 2004.24  4979.5 2002.64  4997.3 2000.04  5000.1 1999.54
  5003.3 2000.04  5021.1 2001.46  5050.0 2001.55  5056.4 2002.19  5064.4 2003.32
  5070.8 2005.12  5085.2 2010.17  5107.4 2013.26  5143.0 2015.97  5207.1 2019.24
  5242.3 2021.55  5292.0 2023.34  5349.7 2026.10  5463.5 2028.81  5490.5 2029.11
#Mann=3,-1,0
  4516.6     0.1       0  4997.3    0.07       0  5003.3     0.1       0
Bank Sta=4997.3,5003.3
Exp/Cntr=0.3,0.1

Type RM Length L Ch R = 1,5045,814,814,814
BEGIN DESCRIPTION:
BANTA BRANCH 11.0
END DESCRIPTION:
XS GIS Cut Line= 2
      2644392.96     10072968.37      2643081.97     10072226.18
#Sta/Elev= 30
  4157.2 2031.74  4172.4 2030.91  4178.2 2031.54  4215.7 2029.49  4221.5 2030.15
  4237.4 2029.05  4259.0 2028.91  4369.2 2024.05  4427.2 2022.70  4537.9 2020.25
  4668.8 2016.98  4889.6 2013.78  4943.1 2012.13  4948.8 2011.77  4964.7 2004.64
  4978.2 1999.69  4992.1 1996.64  4998.2 1996.41  5001.0 1995.91  5004.2 1996.41
  5045.5 1999.63  5081.7 1997.92  5094.5 2001.57  5104.7 2003.41  5132.1 2004.45
  5169.6 2009.37  5219.6 2012.18  5374.5 2017.00  5455.3 2021.43  5663.7 2026.46
#Mann=5,-1,0
  4157.2     0.1       0  4427.2    0.05       0  4537.9     0.1       0
  4998.2    0.07       0  5004.2     0.1       0
Bank Sta=4998.2,5004.2
Exp/Cntr=0.3,0.1

Type RM Length L Ch R = 1,4231,518,518,518
BEGIN DESCRIPTION:
BANTA BRANCH 10.0
END DESCRIPTION:
XS GIS Cut Line= 3
      2644511.04     10072253.12      2643608.23     10071530.87
      2643427.68     10071426.71
#Sta/Elev= 30
  4273.4 2021.14  4390.1 2018.64  4434.3 2016.89  4459.4 2013.94  4488.3 2006.91
  4509.1 2003.75  4531.5 2002.82  4581.1 2003.34  4609.7 2004.94  4637.1 2004.53
  4645.1 2002.72  4651.5 2003.32  4659.5 2001.88  4677.5 2001.58  4857.4 2001.59
  4901.3 2001.98  4936.5 2000.97  4957.3 1997.48  4971.7 1994.22  4979.7 1991.33
  4997.5 1990.05  5000.3 1989.55  5003.5 1990.05  5035.7 1990.38  5093.4 1997.28
  5149.4 2000.39  5235.8 2014.60  5256.6 2015.99  5434.4 2019.31  5638.0 2026.37
#Mann=7,-1,0
  4273.4     0.1       0  4390.1    0.16       0  4434.3     0.1       0
  4677.5    0.16       0  4857.4     0.1       0  4997.5    0.07       0
  5003.5     0.1       0
Bank Sta=4997.5,5003.5
Exp/Cntr=0.3,0.1

Type RM Length L Ch R = 1,3713,482,482,482
BEGIN DESCRIPTION:
BANTA BRANCH 8.0
END DESCRIPTION:
XS GIS Cut Line= 2
      2644622.15     10071787.84      2643942.84     10071129.33
#Sta/Elev= 30
  4505.7 2014.93  4531.2 2014.40  4659.8 2010.58  4695.0 2008.27  4709.2 2006.80
  4730.5 2002.96  4737.5 2002.58  4744.6 2000.55  4751.6 1999.75  4758.8 1997.84
  4772.9 1995.79  4780.8 1995.44  4804.5 1993.59  4822.3 1993.21  4857.8 1993.80
  4907.2 1992.94  4928.6 1991.79  4949.7 1988.36  4989.1 1987.96  4991.9 1987.46
  4995.1 1987.96  5034.6 1988.49  5055.7 1992.97  5069.8 1994.99  5105.3 1999.80
  5176.0 2006.21  5282.0 2009.49  5317.5 2011.27  5416.3 2013.72  5451.8 2015.34
#Mann=7,-1,0
  4505.7     0.1       0  4531.2    0.16       0  4780.8     0.1       0
  4804.5    0.16       0  4989.1    0.07       0  4995.1    0.16       0
  5069.8     0.1       0
Bank Sta=4989.1,4995.1
Exp/Cntr=0.3,0.1

Type RM Length L Ch R = 1,3231,437,437,437
BEGIN DESCRIPTION:
BANTA BRANCH 7.0
END DESCRIPTION:
XS GIS Cut Line= 3
      2644749.13     10071412.77      2644540.79     10071053.38
      2644213.07     10070975.35
#Sta/Elev= 30
  4544.1 2007.46  4609.2 2003.99  4659.4 2001.80  4675.5 2001.56  4712.8 1999.31
  4830.4 1996.99  4836.1 1996.21  4910.7 1992.66  4932.2 1990.87  4938.0 1988.41
  4953.8 1986.42  4956.8 1985.26  4963.3 1985.26  4972.2 1983.39  4983.6 1979.43
  4989.7 1978.46  4992.5 1977.96  4995.7 1978.46  5013.3 1979.01  5020.6 1981.44
  5033.9 1984.31  5044.1 1985.01  5062.7 1988.91  5095.5 1990.61  5167.5 1992.71
  5188.1 1995.33  5194.3 1997.15  5208.6 1999.57  5236.5 2002.82  5296.4 2008.26
#Mann=5,-1,0
  4544.1     0.1       0  4609.2    0.16       0  4659.4     0.1       0
  4989.7    0.07       0  4995.7     0.1       0
Bank Sta=4989.7,4995.7
Exp/Cntr=0.3,0.1

Type RM Length L Ch R = 1,2794,354,354,354
BEGIN DESCRIPTION:
BANTA BRANCH 6.0
END DESCRIPTION:
XS GIS Cut Line= 2
      2645073.51     10071100.32      2644587.39     10070475.31
#Sta/Elev= 30
  4528.9 2009.12  4573.4 2008.08  4635.4 2005.19  4658.4 2003.80  4778.8 1999.53
  4793.3 1998.26  4807.7 1996.36  4815.9 1993.71  4822.2 1992.50  4836.7 1988.14
  4843.0 1986.75  4851.2 1985.64  4892.8 1985.34  4921.8 1984.19  4942.6 1981.74
  4965.2 1981.08  4979.7 1978.98  5003.8 1977.50  5006.6 1977.00  5009.8 1977.50
  5015.0 1979.35  5021.3 1983.27  5035.8 1988.16  5056.7 1991.33  5063.0 1991.81
  5071.1 1993.46  5100.0 1996.56  5120.8 1998.26  5234.9 2004.30  5320.7 2006.34
#Mann=4,-1,0
  4528.9    0.16       0  4635.4     0.1       0  5003.8    0.07       0
  5009.8     0.1       0
Bank Sta=5003.8,5009.8
Exp/Cntr=0.3,0.1

Type RM Length L Ch R = 1,2440,505,505,505
BEGIN DESCRIPTION:
BANTA BRANCH 5.0
END DESCRIPTION:
XS GIS Cut Line= 3
      2645243.90     10070808.56      2644973.08     10070365.88
      2644775.16     10070329.42
#Sta/Elev= 30
  4640.6 2002.47  4720.3 1999.35  4751.2 1996.79  4792.8 1994.95  4851.8 1989.93
  4867.3 1986.89  4873.1 1984.70  4880.7 1982.81  4888.6 1981.79  4931.2 1980.52
  4946.6 1979.58  4967.9 1979.80  4989.2 1977.04  5001.7 1976.46  5004.4 1975.96
  5007.7 1976.46  5033.1 1982.65  5041.4 1983.39  5056.6 1985.80  5068.6 1988.65
  5099.5 1991.90  5126.9 1996.08  5159.6 1999.08  5194.3 2000.37  5215.1 2001.77
  5245.6 2002.58  5276.1 2004.66  5296.4 2004.67  5326.9 2005.70  5360.8 2005.60
#Mann=3,-1,0
  4640.6     0.1       0  5001.7    0.07       0  5007.7     0.1       0
Bank Sta=5001.7,5007.7
Exp/Cntr=0.3,0.1

Type RM Length L Ch R = 1,1935,461,461,461
BEGIN DESCRIPTION:
BANTA BRANCH 4.0
END DESCRIPTION:
XS GIS Cut Line= 3
      2645618.45     10070453.70      2645468.47     10070203.73
      2645218.43     10070053.71
#Sta/Elev= 30
  4691.1 1997.37  4726.0 1994.39  4807.7 1989.88  4831.0 1987.72  4858.2 1982.41
  4866.0 1980.04  4873.8 1976.78  4879.6 1973.01  4886.3 1970.78  4889.1 1970.28
  4892.3 1970.78  4901.0 1972.13  4910.7 1976.63  4916.5 1978.20  4924.3 1978.53
  4947.6 1977.95  4969.0 1975.26  4985.5 1975.71  5005.9 1975.06  5017.6 1977.95
  5027.3 1978.76  5033.1 1980.31  5054.5 1980.94  5091.5 1980.12  5134.2 1980.54
  5143.9 1981.37  5171.1 1988.48  5180.9 1989.74  5208.1 1991.59  5274.2 1997.74
#Mann=3,-1,0
  4691.1     0.1       0  4886.3    0.07       0  4892.3     0.1       0
Bank Sta=4886.3,4892.3
Exp/Cntr=0.3,0.1

Type RM Length L Ch R = 1,1474,330,330,330
BEGIN DESCRIPTION:
BANTA BRANCH 3.0
END DESCRIPTION:
XS GIS Cut Line= 3
      2646018.44     10070153.70      2645868.47     10070003.73
      2645518.45     10069853.72
#Sta/Elev= 30
  4772.9 1998.15  4776.4 1998.15  4801.1 1992.98  4815.3 1990.39  4843.6 1982.21
  4857.7 1979.51  4871.9 1977.93  4886.0 1977.03  4914.3 1976.28  4942.6 1976.09
  4956.7 1975.55  4970.8 1973.23  4981.5 1969.54  4987.7 1969.54  4994.1 1968.07
  4996.5 1966.70  4999.2 1966.20  5002.5 1966.70  5006.8 1966.76  5017.6 1968.72
  5028.5 1970.07  5039.4 1969.63  5052.1 1971.54  5075.7 1972.80  5104.7 1978.30
  5151.8 1981.67  5169.9 1982.14  5199.0 1984.03  5257.0 1986.68  5365.8 1989.95
#Mann=4,-1,0
  4772.9    0.16       0  4801.1     0.1       0  4996.5    0.07       0
  5002.5     0.1       0
Bank Sta=4996.5,5002.5
Exp/Cntr=0.3,0.1

Type RM Length L Ch R = 1,1144,347,347,347
BEGIN DESCRIPTION:
BANTA BRANCH 2.0
END DESCRIPTION:
XS GIS Cut Line= 3
      2646372.09     10069926.69      2645781.84     10069586.43
      2645561.51     10069620.86
#Sta/Elev= 30
  4653.8 2005.55  4761.9 2003.80  4811.8 2000.18  4849.2 1994.78  4870.7 1993.42
  4886.5 1991.49  4923.5 1985.71  4935.4 1982.51  4945.4 1975.85  4951.2 1973.35
  4958.1 1968.32  4981.2 1967.14  4994.3 1965.33  5004.8 1965.43  5025.9 1966.86
  5047.4 1965.95  5050.2 1965.21  5052.9 1964.71  5056.2 1965.21  5062.0 1966.55
  5069.0 1970.06  5074.7 1971.88  5084.7 1973.71  5113.6 1974.18  5133.6 1975.45
  5155.2 1979.81  5224.7 1985.49  5267.2 1987.00  5335.7 1986.83  5558.1 1988.45
#Mann=7,-1,0
  4653.8     0.1       0  5004.8    0.05       0  5050.2    0.07       0
  5056.2    0.05       0  5113.6     0.1       0  5224.7    0.16       0
  5335.7     0.1       0
Bank Sta=5050.2,5056.2
Exp/Cntr=0.3,0.1

Type RM Length L Ch R = 1,797,279,279,279
BEGIN DESCRIPTION:
Mapping XS 50ffb08e
END DESCRIPTION:
XS GIS Cut Line= 4
      2646432.55     10069872.17      2646291.51     10069509.80
      2646146.11     10069399.12      2645572.29     10069583.18
#Sta/Elev= 30
  4525.0 2004.65  4688.8 2002.44  4695.0 2001.98  4713.3 1997.41  4767.7 1993.10
  4822.1 1990.58  4876.5 1989.94  4906.4 1986.65  4911.2 1984.75  4934.3 1980.84
  4942.6 1978.79  4948.9 1975.62  4955.4 1969.64  4963.4 1966.43  4995.8 1960.53
  4998.5 1960.03  5001.8 1960.53  5034.1 1962.83  5042.4 1966.75  5063.2 1970.23
  5178.1 1970.42  5188.5 1972.23  5193.7 1971.54  5209.6 1977.05  5225.8 1979.51
  5333.1 1985.42  5476.4 1986.09  5686.7 1988.11  5693.7 1988.08  5699.2 1988.05
#Mann=7,-1,0
  4525.0     0.1       0  4995.8    0.07       0  5001.8     0.1       0
  5333.1    0.16       0  5476.4     0.1       0  5686.7    0.05       0
  5693.7     0.1       0
Bank Sta=4995.8,5001.8
Exp/Cntr=0.3,0.1

Type RM Length L Ch R = 1,518,175,175,175
BEGIN DESCRIPTION:
Mapping XS 21133b9e
END DESCRIPTION:
XS GIS Cut Line= 4
      2646766.76     10069090.96      2646439.08     10069195.13
      2646265.46     10069227.68      2645472.32     10069585.25
#Sta/Elev= 30
  4560.0 2000.75  4843.5 1991.02  4885.7 1986.52  4898.8 1979.75  4901.5 1977.91
  4906.7 1977.91  4921.6 1966.91  4935.0 1963.70  4955.3 1962.17  4974.1 1958.22
  4982.9 1957.76  4985.6 1957.26  4988.9 1957.76  5016.4 1959.01  5026.6 1961.48
  5031.8 1965.81  5036.9 1963.59  5046.9 1967.10  5057.1 1968.14  5162.9 1969.64
  5277.7 1969.83  5318.5 1971.33  5353.8 1976.13  5384.3 1978.41  5494.2 1984.20
  5495.8 1984.22  5604.7 1984.92  5825.6 1986.95  5932.0 1988.51  5950.5 1988.97
#Mann=12,-1,0
  4560.0     0.1       0  4843.5    0.05       0  4898.8     0.1       0
  4982.9    0.07       0  4988.9     0.1       0  5162.9    0.05       0
  5277.7     0.1       0  5494.2    0.05       0  5495.8    0.16       0
  5604.7     0.1       0  5825.6    0.05       0  5932.0     0.1       0
Bank Sta=4982.9,4988.9
Exp/Cntr=0.3,0.1

Type RM Length L Ch R = 1,343,140,140,140
BEGIN DESCRIPTION:
Mapping XS 4f5becbd
END DESCRIPTION:
XS GIS Cut Line= 4
      2646864.16     10068916.80      2646207.89     10069099.09
      2645574.21     10069356.04      2644932.62     10069732.32
#Sta/Elev= 30
  4507.7 2000.29  4648.5 1998.40  4918.4 1990.91  4939.1 1986.30  4949.5 1980.42
  4959.0 1972.48  4964.2 1970.47  4970.3 1963.58  4980.6 1958.14  4995.4 1955.97
  4998.2 1955.47  5001.4 1955.97  5043.1 1959.69  5063.7 1966.20  5072.1 1967.51
  5263.0 1967.36  5399.7 1970.51  5468.9 1970.31  5525.5 1971.26  5608.7 1971.82
  5614.0 1973.13  5638.1 1971.66  5705.1 1972.58  5742.4 1972.68  6035.9 1974.27
  6287.0 1978.03  6372.0 1979.16  6436.2 1982.07  6580.1 1987.53  6616.4 1988.37
#Mann=10,-1,0
  4507.7     0.1       0  4995.4    0.07       0  5001.4     0.1       0
  5468.9    0.05       0  5525.5     0.1       0  5705.1    0.05       0
  5742.4     0.1       0  6287.0    0.05       0  6436.2     0.1       0
  6580.1    0.05       0
Bank Sta=4995.4,5001.4
Exp/Cntr=0.3,0.1

Type RM Length L Ch R = 1,203,0,0,0
BEGIN DESCRIPTION:
BANTA BRANCH 1.0
END DESCRIPTION:
XS GIS Cut Line= 3
      2646894.83     10068845.73      2646449.93     10068863.10
      2644882.22     10069721.76
#Sta/Elev= 30
  4452.3 1999.29  4475.8 1999.01  4922.0 1990.27  4944.8 1986.37  4956.4 1979.84
  4966.8 1972.37  4972.5 1970.08  4979.0 1963.62  4988.6 1957.81  4998.8 1955.55
  5001.6 1955.05  5004.8 1955.55  5032.3 1957.52  5054.1 1964.00  5097.7 1966.94
  5141.3 1967.07  5157.4 1965.69  5163.1 1966.50  5179.2 1964.80  5304.4 1964.27
  5326.2 1965.79  5342.3 1965.43  5369.8 1967.84  5413.4 1968.92  5745.3 1972.22
  6049.6 1973.75  6356.0 1977.27  6448.6 1979.46  6609.3 1986.17  6685.0 1988.12
#Mann=7,-1,0
  4452.3    0.05       0  4475.8     0.1       0  4998.8    0.07       0
  5004.8     0.1       0  6356.0    0.05       0  6448.6     0.1       0
  6609.3    0.05       0
Bank Sta=4998.8,5004.8
Exp/Cntr=0.3,0.1

Chan Stop Cuts=-1
