--- LEFT BEAR CREEK.prj (project) ---

Proj Title=LEFT BEAR CREEK Base Level Engineering
Current Plan=p01
Default Exp/Contr=0.3,0.1
English Units
Geom File=g01
Flow File=f01
Plan File=p01
Y Axis Title=Elevation
X Axis Title(PF)=Main Channel Distance
X Axis Title(XS)=Station
BEGIN DESCRIPTION:
LEFT BEAR CREEK
END DESCRIPTION:
DSS Export Rating Curves= 0
DSS Export Rating Curve Sorted= 0
DSS Export Volume Flow Curves= 0
DXF OffsetX= 0
DXF OffsetY= 0
DXF ScaleX= 1
DXF ScaleY= 10

--- LEFT BEAR CREEK.p01 (plan) ---

Plan Title=Multiple Run
Short Identifier=Multiple
Geom File=g01
Flow File=f01
Subcritical Flow
K Sum by GR= 0
Std Step Tol= 0.01
Critical Tol= 0.01
Num of Std Step Trials= 20
Max Error Tol= 0.3
Flow Tol Ratio= 0.001
Split Flow NTrial= 30
Split Flow Tol= 0.02
Split Flow Ratio= 0.02
Log Output Level= 0
Friction Slope Method= 1
Unsteady Friction Slope Method= 2
Unsteady Bridges Friction Slope Method= 1
Parabolic Critical Depth
Global Vel Dist=  1 , 1 , 1
Global Log Level= 0
CheckData=True
Encroach Param= -1, 0, 0, 0
BEGIN DESCRIPTION:
Multiple Run
END DESCRIPTION:

--- LEFT BEAR CREEK.f01 (steady flow) ---

Flow Title=Multiple
Program Version=4.10
Number of Profiles= 7
Profile Names=10-year,25-year,50-year,1pct_min,100-year,1pct_plu,500-year
River Rch & RM=LEFT BEAR CREEK,Reach-1         ,32520
     747    1065    1336    1227    1659    2244    2568
River Rch & RM=LEFT BEAR CREEK,Reach-1         ,30344
    1358    2001    2566    2405    3252    4398    5245
River Rch & RM=LEFT BEAR CREEK,Reach-1         ,28063
    1676    2487    3205    3014    4076    5513    6624
River Rch & RM=LEFT BEAR CREEK,Reach-1         ,21474
    2426    3661    4772    4533    6130    8291   10170
River Rch & RM=LEFT BEAR CREEK,Reach-1         ,20604
    2426    3661    4772    4533    6130    8291   10170
River Rch & RM=LEFT BEAR CREEK,Reach-1         ,20190
    2426    3661    4772    4533    6130    8291   10170
River Rch & RM=LEFT BEAR CREEK,Reach-1         ,16143
    2574    3886    5065    4811    6506    8799   10788
River Rch & RM=LEFT BEAR CREEK,Reach-1         ,11365
    3449    5266    6917    6615    8947   12099   15041
River Rch & RM=LEFT BEAR CREEK,Reach-1         ,10361
    3449    5266    6917    6615    8947   12099   15041
River Rch & RM=LEFT BEAR CREEK,Reach-1         ,8541
    3532    5391    7078    6765    9149   12372   15362
Boundary for River Rch & Prof#=LEFT BEAR CREEK,Reach-1         , 1
Up Type= 0
Dn Type= 3
Dn Slope=0.011
Boundary for River Rch & Prof#=LEFT BEAR CREEK,Reach-1         , 2
Up Type= 0
Dn Type= 3
Dn Slope=0.011
Boundary for River Rch & Prof#=LEFT BEAR CREEK,Reach-1         , 3
Up Type= 0
Dn Type= 3
Dn Slope=0.011
Boundary for River Rch & Prof#=LEFT BEAR CREEK,Reach-1         , 4
Up Type= 0
Dn Type= 3
Dn Slope=0.011
Boundary for River Rch & Prof#=LEFT BEAR CREEK,Reach-1         , 5
Up Type= 0
Dn Type= 3
Dn Slope=0.011
Boundary for River Rch & Prof#=LEFT BEAR CREEK,Reach-1         , 6
Up Type= 0
Dn Type= 3
Dn Slope=0.011
Boundary for River Rch & Prof#=LEFT BEAR CREEK,Reach-1         , 7
Up Type= 0
Dn Type= 3
Dn Slope=0.011
DSS Import GetInterval= 0
DSS Import GetPeak= 0
DSS Import FillOption= 0

--- LEFT BEAR CREEK.g01 (geometry) ---

Geom Title=Existing Conditions
Program Version=4.10

River Reach=LEFT BEAR CREEK ,Reach-1
Reach XY= 30
      2743087.66     10008347.22      2744044.42     10008861.85
      2744929.14      10009654.3      2745880.62     10011456.14
      2746374.71     10011570.35      2748648.23     10014588.76
      2748665.34     10015312.44      2747976.59     10016337.14
      2747790.08     10018047.43      2746759.35     10018694.11
      2746017.63     10020140.67      2744659.61     10020036.49
      2744324.23     10020515.64      2743809.26     10020701.07
      2743699.64     10021153.62      2743968.42     10021814.75
      2743672.73      10022211.8      2743259.75     10022240.63
      2742323.88     10021835.97      2742035.46     10022048.61
      2741820.51     10023033.21      2740827.62     10023398.07
      2740923.56      10024079.3      2741276.04     10024373.77
      2740934.61      10024839.4      2738953.89     10024820.92
      2738680.96      10025787.7      2739806.75     10027437.96
       2739522.8       10027876.      2738252.54     10028271.26

Type RM Length L Ch R = 1 ,32520   ,460,460,460
BEGIN DESCRIPTION:
LEFT BEAR CREEK 68.0
END DESCRIPTION:
XS GIS Cut Line= 2
      2743055.84     10009000.81      2743472.48     10008078.99
#Sta/Elev= 30
  4430.4 1969.63  4446.3 1970.23  4474.9 1969.49  4492.5 1969.86  4590.5 1968.96
  4619.1 1967.33  4665.3 1966.11  4723.5 1962.38  4778.4 1960.71  4809.5 1957.78
  4832.6 1958.22  4866.7 1955.36  4899.1 1953.95    4943 1949.24  4959.1 1948.85
    4970 1947.58  4987.7 1944.42  5005.1 1943.75  5051.6 1945.55  5063.7 1945.18
  5085.7 1947.41  5096.6 1947.62  5149.5  1949.8  5195.4 1950.82  5224.3 1952.28
  5276.1 1953.05  5316.1 1954.46    5374 1958.96  5403.9 1962.41    5442  1963.6
#Mann= 3 ,-1 , 0
  4430.4      .1       0  4959.1     .07       0  5096.6      .1       0
Bank Sta=4970,5096.6
XS Rating Curve= 0 ,0
Exp/Cntr=0.3,0.1

Type RM Length L Ch R = 1 ,32060   ,518,518,518
BEGIN DESCRIPTION:
LEFT BEAR CREEK 67.0
END DESCRIPTION:
XS GIS Cut Line= 2
      2743441.25     10009032.08       2743837.1     10008464.35
#Sta/Elev= 30
  4631.4  1955.6  4656.3 1953.64  4706.9 1951.98  4742.7 1948.14  4751.3  1948.2
  4757.5 1949.26  4824.7 1948.04  4858.7 1947.32  4873.2 1945.61  4885.8 1941.97
  4900.6 1940.13    4922 1941.53  4945.1 1941.59    4963 1939.03  4965.8 1938.53
    4969 1939.03  4980.9  1940.2  5001.8 1939.16  5016.7 1940.37  5037.6 1939.57
  5067.3 1940.18  5088.2 1941.52  5094.3 1943.09  5109.1 1944.17    5124 1943.72
  5172.4 1945.48  5192.3 1946.07  5225.2 1947.33  5291.9 1951.59  5323.5 1954.28
#Mann= 7 ,-1 , 0
  4631.4     .05       0  4824.7      .1       0    4963     .07       0
    4969      .1       0  5172.4     .16       0  5192.3      .1       0
  5291.9     .16       0
Bank Sta=4945.1,5088.2
XS Rating Curve= 0 ,0
Exp/Cntr=0.3,0.1

Type RM Length L Ch R = 1 ,31542   ,305,305,305
BEGIN DESCRIPTION:
LEFT BEAR CREEK 66.0
END DESCRIPTION:
XS GIS Cut Line= 3
      2743597.51      10009297.7      2744248.54     10008839.38
        2744285.     10008651.87
#Sta/Elev= 30
  4399.7 1962.61  4446.8 1962.08  4480.7 1959.74  4518.6 1958.49  4533.1 1957.69
  4596.5 1948.98  4682.9 1940.65  4692.1 1939.72  4726.5 1936.54  4791.8 1936.63
  4812.7 1935.86  4816.5 1934.68  4827.5 1933.86  4833.6 1931.27  4839.2 1931.17
  4919.8 1933.43  4970.4 1932.03    4997 1927.18  4999.7 1926.68    5003 1927.18
  5012.3 1927.63  5020.9 1932.04    5027 1938.04  5035.7 1939.91  5157.6 1950.09
  5211.8 1956.24  5232.2 1959.98  5252.6 1960.62  5322.6 1966.51  5386.9 1967.47
#Mann= 9 ,-1 , 0
  4399.7      .1       0  4480.7     .16       0  4518.6      .1       0
  4682.9     .16       0  4692.1      .1       0  4816.5     .16       0
  4839.2      .1       0    4997     .07       0    5003      .1       0
Bank Sta=4970.4,5020.9
XS Rating Curve= 0 ,0
Exp/Cntr=0.3,0.1

Type RM Length L Ch R = 1 ,31237   ,471,471,471
BEGIN DESCRIPTION:
LEFT BEAR CREEK 65.0
END DESCRIPTION:
XS GIS Cut Line= 3
      2743790.22      10009610.2      2744498.54     10008990.42
      2744503.75     10008761.27
#Sta/Elev= 30
  4395.3 1962.33  4433.7 1960.58  4490.6 1959.67  4512.5 1958.09  4547.6 1952.46
  4554.2 1953.18  4567.5 1951.67  4621.2 1946.57  4632.1 1944.98  4646.3 1945.27
    4703 1941.58  4731.7 1938.98  4809.5 1934.54  4879.4 1933.68  4915.8 1932.83
  4958.5 1928.62  4998.3 1924.16    5001 1923.66  5004.3 1924.16  5036.4 1928.01
  5093.3 1929.28  5114.2  1935.2  5142.7 1938.83  5256.6 1944.42  5298.3 1947.53
  5403.2 1951.36  5433.2 1954.64  5473.2 1957.12  5533.2 1963.61  5565.7 1964.04
#Mann= 7 ,-1 , 0
  4395.3      .1       0  4567.5     .16       0  4621.2      .1       0
    4703     .16       0  4879.4      .1       0  4998.3     .07       0
  5004.3      .1       0
Bank Sta=4958.5,5093.3
XS Rating Curve= 0 ,0
Exp/Cntr=0.3,0.1

Type RM Length L Ch R = 1 ,30766   ,422,422,422
BEGIN DESCRIPTION:
LEFT BEAR CREEK 64.0
END DESCRIPTION:
XS GIS Cut Line= 4
       2743988.1     10009797.72      2744540.21      10009667.5
      2744701.66     10009183.13      2744701.66     10009048.26
#Sta/Elev= 30
  4279.2 1954.01  4359.3 1948.37  4462.6 1943.91  4533.7 1940.21  4567.3 1939.82
  4576.1  1938.8  4587.8 1934.92  4615.6 1934.34  4628.9 1937.31  4639.2 1937.59
  4649.5 1935.53  4659.7 1935.22  4665.9 1936.67  4680.3 1936.21  4750.5 1931.08
  4840.3 1926.53  4934.8 1926.13  4951.1 1922.68    4995 1919.71  4997.8 1919.21
    5001 1919.71  5014.3 1921.24  5029.6 1921.23    5046 1923.43  5109.2  1924.3
  5166.7 1923.61  5209.4 1927.34  5235.7 1933.06  5267.3 1935.03  5491.9 1941.11
#Mann= 5 ,-1 , 0
  4279.2      .1       0  4462.6     .16       0  4615.6      .1       0
    4995     .07       0    5001      .1       0
Bank Sta=4951.1,5046
XS Rating Curve= 0 ,0
Exp/Cntr=0.3,0.1

Type RM Length L Ch R = 1 ,30344   ,305,305,305
BEGIN DESCRIPTION:
LEFT BEAR CREEK 63.0
END DESCRIPTION:
XS GIS Cut Line= 2
      2744201.67      10010042.5      2745242.73     10009558.41
#Sta/Elev= 30
    4173 1945.51  4252.6 1941.98    4281 1943.06  4290.8 1941.56  4298.4 1938.03
  4312.8 1934.48  4326.8 1934.79  4356.9    1940  4367.1 1939.76  4395.5 1936.93
  4478.3 1932.63  4566.7  1931.3  4732.4 1922.71  4886.3 1921.38  4898.1 1918.53
  4952.5 1916.07  4993.6 1911.33  4996.3 1910.83  4999.6 1911.33  5012.6 1912.87
  5029.7 1918.45  5035.5 1922.26  5109.6 1930.56  5149.9 1938.42  5195.1 1943.21
  5201.2  1945.2  5229.6 1947.82  5252.5 1947.02  5269.8 1950.99  5321.1 1953.02
#Mann= 3 ,-1 , 0
    4173      .1       0  4993.6     .07       0  4999.6      .1       0
Bank Sta=4898.1,5029.7
XS Rating Curve= 0 ,0
Exp/Cntr=0.3,0.1

Type RM Length L Ch R = 1 ,30039   ,496,496,496
BEGIN DESCRIPTION:
LEFT BEAR CREEK 62.0
END DESCRIPTION:
XS GIS Cut Line= 2
      2744383.98     10010422.69      2745372.07     10009777.83
#Sta/Elev= 30
  4164.4  1933.7    4325 1931.36    4412 1931.23  4514.7 1928.63  4520.7 1929.18
  4535.8    1928  4556.9 1928.49  4608.2 1925.27  4644.4 1924.25    4759 1923.28
  4846.5 1920.12  4874.3 1920.18  4897.9 1918.24  4955.2 1916.31 4965.68 1914.27
  4979.2 1909.95    4982 1909.45  4985.2 1909.95  5027.6 1910.56  5063.8 1913.39
  5069.8 1914.89  5090.8  1922.4  5157.3 1939.03  5178.4 1941.11  5220.6 1947.77
  5256.8 1948.37    5287 1952.77  5320.4 1953.67  5338.3  1954.8  5344.3 1956.38
#Mann= 4 ,-1 , 0
  4164.4      .1       0  4979.2     .07       0  4985.2      .1       0
  5320.4     .05       0
Bank Sta=4965.68,5069.8
XS Rating Curve= 0 ,0
Exp/Cntr=0.3,0.1

Type RM Length L Ch R = 1 ,29543   ,507,507,507
BEGIN DESCRIPTION:
LEFT BEAR CREEK 61.0
END DESCRIPTION:
XS GIS Cut Line= 2
      2744394.36     10010896.68      2745794.44     10010126.37
#Sta/Elev= 30
  3868.8 1942.08  3969.4 1941.28  3985.5 1938.91  4088.7 1934.15  4213.7 1930.72
  4366.2 1924.05  4382.3  1921.1  4429.3 1920.47  4555.7 1917.71  4626.2    1918
  4744.9 1917.36  4856.9  1916.9  4904.1 1915.81  4934.1 1911.11  4938.3 1909.76
  4947.7 1906.88  4964.9 1905.79  4998.6 1903.81  5001.4 1903.31  5004.6 1903.81
  5029.1    1910  5072.7 1924.53  5132.3 1937.89  5149.8 1939.39  5220.3  1944.1
  5257.4 1944.38    5323 1940.92  5382.4 1942.31    5442 1938.85  5466.8 1935.18
#Mann= 11 ,-1 , 0
  3868.8      .1       0  4429.3     .16       0  4555.7     .05       0
  4626.2      .1       0  4744.9     .05       0  4856.9     .16       0
  4934.1     .05       0  4964.9      .1       0  4998.6     .07       0
  5004.6      .1       0  5149.8     .05       0
Bank Sta=4938.3,5029.1
XS Rating Curve= 0 ,0
Exp/Cntr=0.3,0.1

Type RM Length L Ch R = 1 ,29036   ,434,434,434
BEGIN DESCRIPTION:
Mapping XS b75c0ee2
END DESCRIPTION:
XS GIS Cut Line= 3
        2744811.     10011112.83      2745696.46     10010752.57
      2745839.53      10010258.3
#Sta/Elev= 30
  4113.4 1937.14  4248.6 1930.58  4334.3 1928.17  4411.9 1920.75  4491.3 1916.24
  4661.3 1907.41  4715.2 1910.33  4791.9 1909.83  4952.8 1903.84  4997.6 1898.56
  5000.4 1898.06  5003.6 1898.56  5017.5 1899.13  5030.1 1903.37  5039.1 1910.08
  5050.3 1912.58  5094.4 1915.92  5099.6  1914.4    5128 1916.23  5133.2 1913.81
  5161.6 1916.57  5166.8 1914.73  5306.4 1927.56  5345.2 1925.47  5451.2    1931
    5490 1928.33  5495.2 1924.86  5523.6 1925.42  5528.8 1923.18  5583.9 1925.78
#Mann= 6 ,-1 , 0
  4113.4      .1       0  4248.6     .16       0  4491.3      .1       0
  4997.6     .07       0  5003.6      .1       0  5050.3     .05       0
Bank Sta=4952.8,5030.1
XS Rating Curve= 0 ,0
Exp/Cntr=0.3,0.1

Type RM Length L Ch R = 1 ,28602   ,347,347,347
BEGIN DESCRIPTION:
LEFT BEAR CREEK 60.0
END DESCRIPTION:
XS GIS Cut Line= 4
      2745241.01     10011811.94      2745507.41     10011270.73
      2745860.72     10011152.96      2746028.95     10010552.94
#Sta/Elev= 30
  4109.1 1943.75  4150.3 1941.71  4203.5 1938.19  4263.1 1935.96  4396.9 1922.37
  4428.2 1921.64  4552.9  1914.2    4745 1908.64  4787.2 1904.98  4808.3 1901.69
  4813.5 1904.52  4839.9 1905.02  4845.2 1902.51    4861 1901.44    4940 1900.88
  4955.9 1896.76  4971.7 1895.02  4976.8 1895.62    4995    1892  4997.8  1891.5
    5001    1892  5019.1 1893.82 5023.75 1896.46  5040.2 1902.14  5136.5 1901.64
  5218.9 1904.89  5283.3 1904.68  5416.3 1911.73  5666.4 1915.91  5707.9 1916.26
#Mann= 6 ,-1 , 0
  4109.1     .16       0  4150.3      .1       0  4976.8     .05       0
    4995     .04       0    5001     .05       0  5666.4      .1       0
Bank Sta=4955.9,5023.75
XS Rating Curve= 0 ,0
Exp/Cntr=0.3,0.1

Type RM Length L Ch R = 1 ,28255   ,192,192,192
BEGIN DESCRIPTION:
LEFT BEAR CREEK 59.0
END DESCRIPTION:
XS GIS Cut Line= 4
      2745807.45     10012260.53      2745975.68     10011929.68
      2745885.95     10011150.16      2746056.49     10010577.02
#Sta/Elev= 30
  4174.4 1946.74  4344.3 1939.89  4382.3 1939.09  4432.4 1935.41  4476.9 1930.52
  4515.8 1928.21    4538 1925.49  4543.1 1923.72  4560.8 1922.92  4565.8 1924.19
  4611.9 1920.71  4632.1 1916.81  4649.8 1916.92  4654.8 1918.91  4662.3 1918.63
  4822.8 1907.07  4827.8 1907.98  4944.1 1898.34  4964.3 1895.13  4994.5 1888.68
  5002.9 1888.53  5005.6 1888.03  5008.9 1888.53  5044.8 1894.48  5330.2 1900.59
  5426.2 1904.61  5464.6 1903.18  5707.3  1914.1  5848.4 1916.46  5928.2 1918.25
#Mann= 5 ,-1 , 0
  4174.4     .16       0  4344.3     .05       0  5002.9     .04       0
  5008.9     .05       0  5848.4      .1       0
Bank Sta=4964.3,5044.8
XS Rating Curve= 0 ,0
Exp/Cntr=0.3,0.1

Type RM Length L Ch R = 1 ,28063   ,119,119,119
BEGIN DESCRIPTION:
LEFT BEAR CREEK 57.0
END DESCRIPTION:
XS GIS Cut Line= 4
      2746079.42     10012350.33      2746152.34     10012047.45
      2746082.24     10011223.06        2746264.     10010814.79
#Sta/Elev= 30
  4159.6 1933.49  4174.2 1931.85  4179.3 1927.78    4187    1927  4258.1 1925.26
  4361.8 1919.44  4464.7 1917.95    4573 1910.91    4578  1911.8  4692.2 1898.84
  4697.3 1900.35  4715.7 1898.56  4876.3 1896.61  4946.6 1893.67  4966.6 1892.09
  4986.7 1888.04  5003.8 1887.34  5006.5 1886.84  5009.8 1887.34  5044.9 1893.58
    5077 1896.29  5147.3 1895.66  5164.1 1898.92  5169.2 1897.89  5207.5  1900.7
  5302.4 1903.26  5423.7 1911.89    5569 1916.71  5690.6 1923.92  5745.4 1929.47
#Mann= 4 ,-1 , 0
  4159.6     .05       0  5003.8     .04       0  5009.8     .05       0
  5423.7      .1       0
Bank Sta=4946.6,5044.9
XS Rating Curve= 0 ,0
Exp/Cntr=0.3,0.1

Type RM Length L Ch R = 1 ,27944   ,662,662,662
BEGIN DESCRIPTION:
LEFT BEAR CREEK 58.0
END DESCRIPTION:
XS GIS Cut Line= 4
      2746114.86     10012316.37      2746205.14     10012010.82
      2746239.86     10011212.21      2746614.19     10010695.77
#Sta/Elev= 30
  4201.6 1925.93  4264.5 1923.85  4308.6 1920.59  4441.3 1917.26  4496.3 1913.24
  4517.3 1909.99  4627.4 1898.62  4717.5 1895.16    4766 1895.05  4837.6 1894.95
  4887.6 1892.74  4917.7 1891.06  4947.7 1891.31  4994.7 1885.83  4997.5 1885.33
  5000.7 1885.83  5027.8 1889.39  5047.8 1889.93  5067.8 1893.88  5107.8 1893.95
  5137.9  1900.1  5187.9 1904.42    5298  1910.5  5481.7 1917.72    5540 1922.66
  5589.4 1929.03  5661.9 1932.01  5739.2 1941.46  5804.2 1943.26  5957.4 1950.51
#Mann= 4 ,-1 , 0
  4201.6     .05       0    4766      .1       0  4994.7     .07       0
  5000.7      .1       0
Bank Sta=4887.6,5067.8
XS Rating Curve= 0 ,0
Exp/Cntr=0.3,0.1

Type RM Length L Ch R = 1 ,27282   ,518,518,518
BEGIN DESCRIPTION:
LEFT BEAR CREEK 56.0
END DESCRIPTION:
XS GIS Cut Line= 2
      2746183.46     10012364.53      2747441.79     10011288.44
#Sta/Elev= 30
  4417.6 1923.97    4500 1917.53  4602.5 1913.28  4698.7 1908.56  4754.7 1896.76
  4762.1 1897.51  4811.8 1892.21  4891.2 1889.03  4918.2  1886.6  4961.1 1885.77
  4986.6 1880.88  4989.4 1880.38  4992.6 1880.88    5017 1881.63  5031.3 1886.61
  5045.6  1890.5  5074.1 1893.28  5199.2 1894.68  5258.5 1897.32    5365 1898.66
  5466.8 1904.99  5535.8 1912.83  5563.7 1916.02  5613.1 1924.87  5676.8 1930.85
    5713 1937.38  5746.7 1940.22  5783.3 1940.92  6006.4 1953.03  6073.3 1956.61
#Mann= 11 ,-1 , 0
  4417.6     .05       0  4602.5      .1       0  4762.1     .05       0
  4891.2      .1       0  4986.6     .07       0  4992.6      .1       0
  5199.2     .05       0  5466.8      .1       0  5535.8     .16       0
  5746.7      .1       0  6006.4     .05       0
Bank Sta=4961.1,5031.3
XS Rating Curve= 0 ,0
Exp/Cntr=0.3,0.1

Type RM Length L Ch R = 1 ,26764   ,454,454,454
BEGIN DESCRIPTION:
LEFT BEAR CREEK 55.0
END DESCRIPTION:
XS GIS Cut Line= 3
      2746365.73     10012750.84      2746838.82      10012499.1
      2747889.13     10011470.49
#Sta/Elev= 30
  4239.7  1917.9  4388.8 1909.41  4482.3 1906.62    4551 1900.22  4602.8 1894.88
  4670.3 1893.97  4703.9 1893.49  4901.3 1885.18  4948.8 1879.34  4980.7 1874.07
  4995.4 1872.58  4998.2 1872.08  5001.4 1872.58  5012.6 1872.75  5047.9  1879.4
  5083.1 1886.02  5125.6 1885.42  5153.9 1888.32  5219.7 1888.72    5260 1891.56
  5292.7  1890.8    5364 1894.32  5427.3 1898.02  5508.2 1907.43  5755.1  1922.4
    6052 1931.72  6087.4 1929.95  6136.8 1930.91  6172.3 1936.99  6245.7 1940.42
#Mann= 14 ,-1 , 0
  4239.7     .05       0    4551      .1       0  4670.3     .05       0
  4703.9      .1       0  4901.3     .05       0  4980.7      .1       0
  4995.4     .07       0  5001.4      .1       0  5219.7     .05       0
  5292.7      .1       0    5364     .05       0  5427.3      .1       0
  5508.2     .16       0  5755.1      .1       0
Bank Sta=4948.8,5047.9
XS Rating Curve= 0 ,0
Exp/Cntr=0.3,0.1

Type RM Length L Ch R = 1 ,26310   ,362,362,362
BEGIN DESCRIPTION:
LEFT BEAR CREEK 54.0
END DESCRIPTION:
XS GIS Cut Line= 3
      2746465.54     10013076.36      2747242.46      10012724.8
      2748282.82     10011758.13
#Sta/Elev= 30
  4072.7 1915.33  4091.8 1913.75  4108.8 1906.82  4114.9 1902.35    4138 1896.08
  4360.8 1892.24  4438.1 1891.18    4622  1883.6  4789.3 1880.96  4892.7 1881.22
  4925.5  1875.4  4937.4 1873.78  4962.3  1874.9  4987.3 1868.84  4998.5 1868.44
  5001.2 1867.94  5004.5 1868.44  5043.5 1870.55  5057.6 1875.08    5065 1879.85
  5071.8 1881.94  5138.4 1883.26  5319.5 1889.74  5347.9 1892.46  5439.7  1906.9
  5595.6  1916.7  5758.3 1921.41  5991.9 1922.22  6225.4 1925.54  6345.6 1931.88
#Mann= 6 ,-1 , 0
  4072.7     .05       0  4360.8      .1       0  4962.3     .16       0
  4998.5     .07       0  5004.5     .16       0  5138.4      .1       0
Bank Sta=4925.5,5057.6
XS Rating Curve= 0 ,0
Exp/Cntr=0.3,0.1

Type RM Length L Ch R = 1 ,25948   ,476,476,476
BEGIN DESCRIPTION:
LEFT BEAR CREEK 53.0
END DESCRIPTION:
XS GIS Cut Line= 2
      2746664.33      10013371.5      2748834.84     10012325.28
#Sta/Elev= 30
  4123.1 1915.39  4260.9 1907.73  4317.8  1899.3    4448 1887.07  4611.9 1882.58
  4904.8 1879.33  4933.1 1871.56  4949.2 1869.15  5052.7 1869.39  5072.3 1866.89
    5075 1866.39  5078.3 1866.89  5092.3 1869.83    5115 1877.89  5135.1 1877.96
  5181.7 1878.81    5211 1881.08  5293.5  1881.4  5405.4 1886.79  5448.7 1892.04
  5517.2 1895.49  5856.2 1910.39    5974 1917.65  6036.3 1924.17  6137.8 1929.64
  6200.1 1937.51  6300.2 1940.25    6365 1942.21  6416.7  1944.5  6532.6 1947.31
#Mann= 13 ,-1 , 0
  4123.1     .05       0  4933.1      .1       0  5072.3     .07       0
  5078.3      .1       0  5135.1     .16       0  5181.7     .05       0
  5293.5      .1       0  5405.4     .05       0  5517.2      .1       0
  5856.2     .16       0  6300.2     .05       0    6365      .1       0
  6416.7     .05       0
Bank Sta=4933.1,5092.3
XS Rating Curve= 0 ,0
Exp/Cntr=0.3,0.1

Type RM Length L Ch R = 1 ,25472   ,460,460,460
BEGIN DESCRIPTION:
LEFT BEAR CREEK 52.0
END DESCRIPTION:
XS GIS Cut Line= 2
      2747081.03      10013762.1      2748633.05     10012809.02
#Sta/Elev= 30
  4239.8 1911.84  4246.3 1910.97  4265.7 1909.34    4345 1896.96    4403 1883.57
  4436.3 1879.85  4541.9 1876.55  4640.3 1875.83  4687.2 1876.31  4797.3  1873.5
  4866.9 1875.68  4940.9 1867.81  4961.4  1863.6  4996.6 1861.36  4999.3 1860.86
  5002.6 1861.36    5023 1865.73  5044.7 1865.93  5058.2 1868.35  5093.4 1882.57
  5199.3 1888.82  5218.1 1890.22  5318.3 1895.41  5398.6 1899.23  5545.5 1911.63
  5609.4 1912.81    5794 1918.95  5850.9 1924.65  5966.9 1928.22  6061.1 1937.69
#Mann= 13 ,-1 , 0
  4239.8     .05       0  4246.3      .1       0  4436.3     .05       0
  4640.3      .1       0  4866.9     .05       0  4961.4      .1       0
  4996.6     .07       0  5002.6      .1       0  5199.3     .16       0
  5218.1      .1       0  5318.3     .16       0  5609.4      .1       0
    5794     .16       0
Bank Sta=4940.9,5058.2
XS Rating Curve= 0 ,0
Exp/Cntr=0.3,0.1

Type RM Length L Ch R = 1 ,25012   ,354,354,354
BEGIN DESCRIPTION:
LEFT BEAR CREEK 51.0
END DESCRIPTION:
XS GIS Cut Line= 3
       2747117.5     10013861.08      2747690.38     10013907.96
      2748714.83     10013299.52
#Sta/Elev= 30
  4161.6 1910.99  4197.1 1907.39  4251.6 1899.53  4313.1 1894.77  4373.1    1882
    4378 1882.46  4403.4 1877.07  4439.5 1875.24  4626.2 1873.64  4704.4 1870.52
  4912.8    1872  4955.6 1865.04  4978.4 1860.14  4998.7 1858.15  5001.4 1857.65
  5004.7 1858.15  5023.9 1860.46  5036.6 1864.69  5051.1 1868.81  5082.1 1873.32
    5187 1876.62  5236.4 1880.51  5279.1 1884.33  5304.8 1888.54  5380.4 1896.75
    5416 1903.04  5444.7 1908.42  5574.2 1923.93    5746 1939.39  5927.9 1943.76
#Mann= 12 ,-1 , 0
  4161.6     .05       0  4197.1      .1       0    4378     .05       0
  4439.5      .1       0  4998.7     .07       0  5004.7      .1       0
  5082.1     .16       0    5187      .1       0  5236.4     .05       0
  5304.8      .1       0    5416     .16       0  5574.2      .1       0
Bank Sta=4955.6,5036.6
XS Rating Curve= 0 ,0
Exp/Cntr=0.3,0.1

Type RM Length L Ch R = 1 ,24658   ,783,783,783
BEGIN DESCRIPTION:
LEFT BEAR CREEK 50.0
END DESCRIPTION:
XS GIS Cut Line= 4
      2747153.93     10014215.25      2747789.34     10014225.66
      2748607.05     10013819.41      2749153.42     10013418.74
#Sta/Elev= 30
  4001.2 1909.04  4075.7 1901.95  4155.8 1898.41  4213.4  1892.6  4295.8 1885.28
  4395.8 1880.95  4447.5    1877  4467.7 1875.68  4697.2 1868.48  4780.9 1868.55
  4847.9 1870.64  4959.5  1862.6  5001.2 1854.51    5004 1854.01  5007.2 1854.51
  5048.9  1862.8  5061.2 1867.86  5071.2 1868.61  5163.9 1867.93  5302.1  1869.5
  5369.3 1872.57  5406.2 1879.87  5444.2 1893.43  5486.9  1906.9  5501.6 1909.86
  5652.1 1922.67  5740.3 1927.76  5855.3 1929.57  6026.7 1930.37  6227.3 1928.61
#Mann= 10 ,-1 , 0
  4001.2     .05       0  4213.4      .1       0  4447.5     .05       0
  4467.7      .1       0  5001.2     .07       0  5007.2      .1       0
  5163.9     .05       0  5444.2      .1       0  5501.6     .16       0
  5652.1      .1       0
Bank Sta=4959.5,5048.9
XS Rating Curve= 0 ,0
Exp/Cntr=0.3,0.1

Type RM Length L Ch R = 1 ,23875   ,350,350,350
BEGIN DESCRIPTION:
LEFT BEAR CREEK 49.0
END DESCRIPTION:
XS GIS Cut Line= 4
        2747555.     10014418.38      2748487.25     10014673.58
      2748971.63     10014491.29      2749543.97     10013830.49
#Sta/Elev= 30
  3851.1 1881.35  4279.8    1872    4346 1872.27  4454.6 1866.64  4549.3 1864.58
  4872.4 1864.83  4904.4 1858.45  4933.6 1857.33  4948.7 1856.07  4968.8 1850.91
  4995.5 1847.15  4998.3 1846.65  5001.5 1847.15  5011.3 1847.56 5018.75 1857.15
  5028.7 1873.58  5043.3 1880.79  5138.9 1897.39  5226.6 1909.36  5371.3 1915.94
  5427.3 1918.51  5479.4 1919.59    5586 1921.61  5730.3 1923.62  5744.6 1923.41
  5933.8 1924.41    6016 1921.21  6083.2 1917.07  6132.3 1923.22  6209.4 1928.01
#Mann= 14 ,-1 , 0
  3851.1     .05       0  4933.6      .1       0  4968.8     .16       0
  4995.5     .07       0  5001.5     .16       0  5226.6      .1       0
  5371.3     .16       0  5427.3      .1       0  5479.4     .05       0
    5586      .1       0  5730.3     .16       0  5744.6      .1       0
    6016     .05       0  6083.2      .1       0
Bank Sta=4933.6,5018.75
XS Rating Curve= 0 ,0
Exp/Cntr=0.3,0.1

Type RM Length L Ch R = 1 ,23525   ,449,449,449
BEGIN DESCRIPTION:
LEFT BEAR CREEK 48.0
END DESCRIPTION:
XS GIS Cut Line= 3
      2747601.85     10014678.79      2748627.88     10014949.62
      2749258.09     10014944.41
#Sta/Elev= 30
  3838.8 1881.83  3977.2 1877.49  4030.6 1877.46  4070.8 1874.42  4124.9 1874.83
  4201.9 1871.34  4264.4 1871.48    4280 1872.28  4455.8 1863.42    4549 1862.55
  4578.9 1863.79  4794.2 1859.15  4902.8 1858.23  4920.6 1854.71  4960.6 1852.28
  4985.1 1846.88  4987.6 1846.03  4990.3 1845.53  4993.6 1846.03  5011.6 1846.87
  5020.6 1852.68 5023.18 1855.52  5030.6 1862.09  5040.6 1867.43  5060.6 1873.68
  5182.5 1905.11  5220.6 1915.19  5260.6 1920.32  5430.6 1930.99  5530.2 1939.01
#Mann= 9 ,-1 , 0
  3838.8      .1       0  3977.2     .05       0  4201.9      .1       0
  4264.4     .05       0  4794.2      .1       0  4985.1     .16       0
  4987.6     .07       0  4993.6     .16       0  5182.5      .1       0
Bank Sta=4920.6,5023.18
XS Rating Curve= 0 ,0
Exp/Cntr=0.3,0.1

Type RM Length L Ch R = 1 ,23076   ,306,306,306
BEGIN DESCRIPTION:
LEFT BEAR CREEK 47.0
END DESCRIPTION:
XS GIS Cut Line= 2
      2747575.83     10015022.55      2748987.21     10015501.69
#Sta/Elev= 30
  3880.8 1883.44  3894.4 1883.14  3957.2 1880.25  4088.1 1877.79  4356.2 1868.84
  4435.5 1866.22  4485.5 1865.51  4705.4 1857.52  4862.4 1855.18  4893.8  1853.4
  4939.6 1851.91    4975 1846.13    5000 1844.64  5002.8 1844.14    5006 1844.64
  5013.6 1848.33 5018.18 1853.64    5019 1856.12  5034.7 1867.73  5045.2 1872.58
  5050.8 1877.18  5082.2 1889.81  5087.5 1893.15  5108.3 1898.36  5150.9 1902.93
  5171.1 1907.12  5176.4  1906.6  5193.1 1910.39  5214.2  1913.1  5371.3 1921.72
#Mann= 8 ,-1 , 0
  3880.8     .05       0  3894.4      .1       0  4356.2     .05       0
  4435.5      .1       0    4975     .16       0    5000     .07       0
    5006     .16       0    5019      .1       0
Bank Sta=4893.8,5018.18
XS Rating Curve= 0 ,0
Exp/Cntr=0.3,0.1

Type RM Length L Ch R = 1 ,22770   ,428,428,428
BEGIN DESCRIPTION:
LEFT BEAR CREEK 46.0
END DESCRIPTION:
XS GIS Cut Line= 2
      2747815.38     10015288.16      2748768.47     10015793.35
#Sta/Elev= 30
  4210.2 1874.61  4265.5 1872.96  4417.4 1868.65  4429.7 1867.79    4468 1860.65
  4484.3 1861.28    4512 1859.08  4666.4 1856.09  4720.6 1856.78  4846.9 1854.71
  4868.9 1851.68  4910.1  1849.9  4949.4 1849.81  4991.6 1844.27  4994.4 1843.77
  4997.6 1844.27  5017.2 1845.87  5028.6  1850.6  5044.2 1856.88  5051.2  1863.1
  5061.2  1867.4  5083.2 1874.03  5088.9 1874.31  5105.2 1880.02  5110.8 1879.86
  5127.2 1883.94  5193.2 1892.77  5215.2  1893.9  5253.5 1899.08  5288.9 1901.09
#Mann= 5 ,-1 , 0
  4210.2     .05       0  4265.5      .1       0  4910.1     .16       0
  4991.6     .07       0  4997.6     .16       0
Bank Sta=4868.9,5028.6
XS Rating Curve= 0 ,0
Exp/Cntr=0.3,0.1

Type RM Length L Ch R = 1 ,22342   ,362,362,362
BEGIN DESCRIPTION:
LEFT BEAR CREEK 45.0
END DESCRIPTION:
XS GIS Cut Line= 3
       2747534.1     10015470.44      2748409.13     10016095.46
      2748778.95     10015965.24
#Sta/Elev= 30
    4151 1886.56  4241.7 1881.55  4371.6  1874.2  4493.2 1870.04  4579.3  1859.1
    4594 1859.14  4629.6 1855.77  4721.8  1853.3  4751.3 1854.74  4837.3 1854.71
  4866.8 1849.04  4893.9 1846.22  4919.6 1845.59  5013.6 1844.39  5016.3 1843.89
  5019.6 1844.39  5053.5 1844.95  5059.8 1846.55  5065.9 1849.73  5074.5 1852.49
  5080.7 1853.02  5099.8 1851.86  5151.9 1851.06  5228.6 1854.02  5336.9 1859.32
  5393.6  1864.3  5460.7 1873.88  5517.4 1885.16    5574 1889.27  5618.4    1894
#Mann= 7 ,-1 , 0
    4151     .05       0  4241.7      .1       0  4919.6     .16       0
  5013.6     .07       0  5019.6     .16       0  5099.8      .1       0
  5393.6     .16       0
Bank Sta=4866.8,5065.9
XS Rating Curve= 0 ,0
Exp/Cntr=0.3,0.1

Type RM Length L Ch R = 1 ,21980   ,506,506,506
BEGIN DESCRIPTION:
LEFT BEAR CREEK 44.0
END DESCRIPTION:
XS GIS Cut Line= 3
      2747237.24     10015965.24       2748268.5     10016345.46
      2748824.62      10016059.6
#Sta/Elev= 30
  4167.1 1901.14  4193.9 1898.53    4243 1892.76  4322.3 1889.17  4377.9 1880.12
  4438.8    1880  4494.3 1874.25  4641.2 1867.37  4650.6 1865.16    4680 1856.47
  4797.2 1850.79  4874.1 1851.29  4893.2 1850.15  4899.2 1847.92  4924.3 1844.54
  4969.3 1844.45  5037.7 1844.09  5040.5 1843.59  5043.7 1844.09  5047.9 1844.25
  5071.2 1844.86  5095.7 1848.58  5106.9 1851.23  5138.3  1849.6  5348.5 1849.07
  5594.1 1859.43  5631.3 1861.65  5692.2 1868.67  5803.1 1886.79  5891.5 1892.38
#Mann= 8 ,-1 , 0
  4167.1      .1       0  4193.9     .05       0  4650.6      .1       0
  4969.3     .05       0  5037.7    .033       0  5043.7     .05       0
  5047.9      .1       0  5594.1     .16       0
Bank Sta=4899.2,5095.7
XS Rating Curve= 0 ,0
Exp/Cntr=0.3,0.1

Type RM Length L Ch R = 1 ,21474   ,74,74,74
BEGIN DESCRIPTION:
Mapping XS f0c7f284
END DESCRIPTION:
XS GIS Cut Line= 4
      2747179.39     10016622.16      2747752.32     10016679.45
      2747981.49     10016781.01      2748674.25     10017063.25
#Sta/Elev= 30
  4278.7 1904.53  4343.9 1898.47    4349 1899.33  4438.6 1889.52  4449.5 1887.87
  4468.7 1882.62    4519 1873.63  4544.9 1865.87  4579.3 1862.21  4629.5 1862.38
  4659.7 1859.65  4770.2 1853.73  4800.4 1849.48  4854.5 1847.65  4861.2 1846.87
    4872 1845.05  4900.8 1844.17  5080.1 1844.31  5112.7 1845.73  5234.2 1844.87
  5335.8 1846.87  5341.2 1846.98  5365.3  1845.6  5389.1 1839.46  5425.8 1843.42
  5468.6 1843.64  5597.9 1845.78  5710.3 1846.23  5810.8 1848.56  5853.2  1849.3
#Mann= 6 ,-1 , 0
  4278.7      .1       0  4854.5     .07       0  5335.8      .1       0
  5468.6     .16       0  5597.9      .1       0  5810.8     .05       0
Bank Sta=4861.2,5341.2
XS Rating Curve= 0 ,0
Exp/Cntr=0.3,0.1

Type RM Length L Ch R = 1 ,21400   ,76,76,76
BEGIN DESCRIPTION:
Mapping XS 3c0bdf25
END DESCRIPTION:
XS GIS Cut Line= 4
      2747237.27     10016697.02      2747729.44     10016762.12
      2748000.27     10016855.87      2748633.28     10017113.01
#Sta/Elev= 30
    4353 1906.84  4367.7 1906.21  4435.9 1893.65  4465.2 1888.92  4495.4 1880.56
  4519.6 1876.89    4593 1859.51  4656.8 1859.85    4677 1857.32  4757.7 1852.89
  4767.8 1852.28    4798 1847.99  4828.5 1846.99  4872.3 1848.42  4898.1 1853.77
  4929.3 1854.12  4934.6 1852.26  4960.5 1854.12  5085.1 1852.46  5141.6 1844.69
    5296 1845.75  5331.7 1846.32    5350 1845.21  5361.2 1841.63  5379.6 1839.26
  5409.4 1843.26  5425.5 1843.34  5564.6 1844.93  5677.1 1845.52  5819.3 1849.12
#Mann= 8 ,-1 , 0
    4353      .1       0  4435.9     .05       0  4757.7     .07       0
  5085.1     .16       0    5296      .1       0  5425.5     .16       0
  5564.6      .1       0  5819.3     .05       0
Bank Sta=4767.8,5331.7
XS Rating Curve= 0 ,0
Exp/Cntr=0.3,0.1

Type RM Length L Ch R = 1 ,21324   ,138,138,138
BEGIN DESCRIPTION:
Mapping XS d612bedc
END DESCRIPTION:
XS GIS Cut Line= 4
      2747252.29     10016783.61      2747705.45     10016830.49
      2747997.11     10016937.26      2748610.68      10017170.3
#Sta/Elev= 30
  4385.2 1909.71  4430.8 1900.72  4435.8 1901.26  4529.6 1876.74  4628.5 1857.35
    4683 1857.43  4703.1 1854.78  4833.8 1846.58  4867.7 1847.63  4886.6 1850.72
  4918.1 1843.26  4953.9 1839.05  4961.1 1836.07  4984.4 1830.93  5003.5 1830.25
  5040.1  1833.2  5046.3 1835.82    5057 1839.04  5070.7 1843.18  5101.2 1845.03
  5120.9 1848.61  5126.4 1846.37  5149.1 1844.05  5326.9 1846.19  5360.2 1839.87
  5381.8 1839.68  5398.8  1842.9  5476.2 1843.13  5758.5 1847.21  5807.7 1848.66
#Mann= 7 ,-1 , 0
  4385.2     .16       0  4953.9     .07       0    5057     .16       0
  5149.1      .1       0  5360.2     .16       0  5476.2      .1       0
  5758.5     .05       0
Bank Sta=4961.1,5046.3
XS Rating Curve= 0 ,0
Exp/Cntr=0.3,0.1

Type RM Length L Ch R = 1 ,21186   ,582,582,582
BEGIN DESCRIPTION:
LEFT BEAR CREEK 43.0
END DESCRIPTION:
XS GIS Cut Line= 4
      2747287.18     10016820.29       2748120.5     10017132.78
      2748446.02     10017215.25      2748858.35     10017727.41
#Sta/Elev= 30
  4444.8 1904.81  4495.8 1892.71    4526 1888.44    4551 1879.68  4581.2 1872.33
  4611.5 1867.87  4666.7 1855.34  4727.2  1855.5  4837.5 1846.73  4928.3 1846.11
  4958.8 1839.23 4963.07 1837.51  4978.2 1831.32  5008.2  1830.1  5054.9  1837.6
  5063.6 1838.04  5093.9 1839.78  5108.3 1838.36  5154.4 1843.65  5239.8 1843.15
  5325.3 1845.76  5353.3 1840.22  5394.6 1839.62  5841.9 1846.96  5870.7    1846
  5891.5 1838.58  5899.5 1838.26  5941.1 1848.12  6054.7 1860.69  6328.1 1885.53
#Mann= 4 ,-1 , 0
  4444.8      .1       0  4958.8     .07       0  5063.6     .16       0
  6328.1      .1       0
#XS Ineff= 2 ,-1
  5326.7 5792.61 1845.62 5862.22 5978.69 1847.22
Permanent Ineff=
       F       F
Bank Sta=4963.07,5054.9
XS Rating Curve= 0 ,0
Exp/Cntr=0.3,0.1

Type RM Length L Ch R = 1 ,20604   ,414,414,414
BEGIN DESCRIPTION:
LEFT BEAR CREEK 42.0
END DESCRIPTION:
XS GIS Cut Line= 4
      2747593.09      10017069.1      2747732.31     10017568.85
      2748167.81     10017779.46      2748749.64     10018018.62
#Sta/Elev= 30
  4420.8 1849.97  4560.6 1846.45  4581.3 1843.91  4607.9 1846.86  4868.1  1844.5
  4902.3  1843.8  4907.5 1841.13  4939.5 1839.99  4946.4 1835.54  4968.6 1831.17
  5024.2 1830.66  5075.6 1835.57  5120.8 1838.06  5171.6  1836.9  5188.6  1832.9
  5223.9 1830.12  5284.5 1832.92  5301.6 1835.98  5327.1 1835.69  5380.5 1835.18
  5449.4 1838.06  5497.3 1842.21  5557.3  1852.3  5662.1  1862.4  5681.3 1861.43
  5734.2 1864.63  5766.9 1867.61  5898.2 1875.86  5943.5 1878.84  6052.4 1888.15
#Mann= 10 ,-1 , 0
  4420.8     .16       0  4939.5     .07       0  5075.6     .16       0
  5327.1      .1       0  5557.3     .05       0  5662.1      .1       0
  5734.2     .05       0  5766.9      .1       0  5898.2     .05       0
  5943.5      .1       0
Bank Sta=4946.4,5075.6
XS Rating Curve= 0 ,0
Exp/Cntr=0.3,0.1

Type RM Length L Ch R = 1 ,20190   ,211,211,211
BEGIN DESCRIPTION:
Mapping XS 19d416eb
END DESCRIPTION:
XS GIS Cut Line= 4
      2747657.35     10017515.32      2747707.32     10017882.99
      2748260.62     10018207.82      2748628.31      10018293.5
#Sta/Elev= 30
  4479.2 1845.23  4618.9 1839.86  4673.8 1838.62  4751.2 1837.33  4818.6  1837.8
  4909.6 1836.52  4932.7 1834.79  4939.6 1832.56  4950.7 1831.75  4982.5 1830.57
  5071.9 1831.19  5121.2 1830.85  5136.6 1829.79  5139.9 1830.29  5160.9 1832.62
  5222.8  1841.2  5281.4 1847.51  5291.3 1849.21  5297.1 1851.74  5318.5 1853.81
  5334.2  1857.2  5396.9 1858.81  5441.8 1861.18  5457.3  1862.3  5510.2 1863.11
  5628.2  1868.1    5695 1872.07  5718.4 1872.38  5797.7 1878.25  5869.4 1886.87
#Mann= 7 ,-1 , 0
  4479.2     .05       0  4950.7     .16       0  4982.5     .07       0
  5139.9     .16       0  5160.9      .1       0  5396.9     .05       0
  5441.8      .1       0
Bank Sta=4939.6,5160.9
XS Rating Curve= 0 ,0
Exp/Cntr=0.3,0.1

Type RM Length L Ch R = 1 ,19979   ,157,157,157
BEGIN DESCRIPTION:
LEFT BEAR CREEK 41.0
END DESCRIPTION:
XS GIS Cut Line= 3
       2747639.5     10017486.72      2747735.88     10018354.18
      2748439.09     10018611.19
#Sta/Elev= 30
  4364.9 1845.56  4580.1 1838.95  4824.7 1836.69  4915.3 1832.52  4942.3 1829.06
  4965.6 1823.88  5012.9 1822.02  5015.6 1821.52  5018.9 1822.02    5026 1822.68
  5032.9 1825.18  5037.9 1828.49  5046.1 1836.47  5056.1 1841.83  5066.2 1843.35
  5128.4 1845.66  5156.8 1845.63  5186.9 1843.67  5207.1 1847.15  5253.7 1848.34
  5325.6 1853.48  5503.4 1856.11  5659.9 1858.67  5857.7 1865.81    5863 1864.96
  5888.2 1866.24  5893.5 1864.98  5924.1 1864.22  5949.3 1865.15  5986.4 1864.38
#Mann= 4 ,-1 , 0
  4364.9     .05       0  5012.9     .04       0  5018.9     .05       0
  5503.4      .1       0
Bank Sta=4942.3,5037.9
XS Rating Curve= 0 ,0
Exp/Cntr=0.3,0.1

Type RM Length L Ch R = 1 ,19822   ,262,262,262
BEGIN DESCRIPTION:
LEFT BEAR CREEK 40.0
END DESCRIPTION:
XS GIS Cut Line= 4
      2747318.24     10017251.16      2747500.28     10017508.17
      2747593.09     10018514.82      2747778.71     10019046.69
#Sta/Elev= 30
  4024.2 1864.92  4032.9 1864.03  4063.9 1859.68  4125.6 1853.18  4162.1    1853
  4220.4 1849.04  4284.7 1848.52  4481.5 1840.18  4856.9 1835.51  4920.3 1830.87
  4927.2 1828.63  4994.5 1820.59  4997.2 1820.09  5000.5 1820.59    5025 1820.87
  5087.9 1827.88  5139.7 1834.64  5258.6 1837.58    5347  1834.9  5445.9 1834.56
  5502.7 1830.04  5518.4 1830.08  5528.5 1832.29  5533.8 1830.53  5539.6  1833.3
  5559.5 1837.68  5564.8 1837.04  5621.7 1843.59  5714.9 1851.24  5913.4 1861.13
#Mann= 5 ,-1 , 0
  4024.2     .16       0  4032.9      .1       0  4063.9     .05       0
  4994.5     .04       0  5000.5     .05       0
Bank Sta=4927.2,5087.9
XS Rating Curve= 0 ,0
Exp/Cntr=0.3,0.1

Type RM Length L Ch R = 1 ,19560   ,459,459,459
BEGIN DESCRIPTION:
LEFT BEAR CREEK 39.0
END DESCRIPTION:
XS GIS Cut Line= 4
      2746943.43     10017393.98      2747186.15     10018082.89
      2747503.85      10018539.8      2747735.38     10019059.86
#Sta/Elev= 30
  4012.5 1879.19  4217.2 1856.99    4283 1848.63  4362.1 1841.17  4375.9 1842.03
  4401.5 1839.32  4637.8  1833.1    4896 1833.53  4952.8    1828  4955.7 1827.66
  4967.6 1826.32  4988.5 1820.55  5000.4 1819.63  5003.1 1819.13  5006.4 1819.63
  5047.9 1820.67    5075 1824.76  5110.8 1827.85  5182.4 1831.35  5314.7 1832.27
  5391.3 1827.79  5396.8 1829.97  5402.3 1828.86    5420  1833.2    5525 1842.94
  5555.5 1846.05  5593.7    1847  5669.1 1853.75    5784 1857.79  5868.7 1861.23
#Mann= 8 ,-1 , 0
  4012.5     .16       0  4217.2      .1       0  4955.7     .16       0
  5000.4     .07       0  5006.4     .16       0    5525      .1       0
  5669.1     .05       0    5784      .1       0
Bank Sta=4952.8,5110.8
XS Rating Curve= 0 ,0
Exp/Cntr=0.3,0.1

Type RM Length L Ch R = 1 ,19101   ,300,300,300
BEGIN DESCRIPTION:
LEFT BEAR CREEK 38.0
END DESCRIPTION:
XS GIS Cut Line= 4
      2746353.17     10018033.85      2746769.81     10018360.21
      2747106.61     10018707.43      2747662.14      10019134.5
#Sta/Elev= 30
  4191.9 1850.76  4231.3  1848.3  4281.1 1848.26    4310  1845.6    4395 1844.77
  4423.9 1842.18  4892.5 1834.05  4920.8 1832.57    4935 1829.78    4949 1824.77
  4970.2 1818.27  5002.5 1817.63  5005.2 1817.13  5008.5 1817.63  5062.1  1820.5
  5083.4 1825.01  5097.5 1826.26    5140 1825.06  5210.3  1825.9  5324.5 1830.49
  5374.3 1834.02  5396.4 1839.87  5459.5 1848.72  5538.3 1851.12  5581.9 1854.77
  5641.5  1855.1  5702.3 1858.16  5766.7 1858.26  5882.3 1861.38  5905.6 1862.37
#Mann= 5 ,-1 , 0
  4191.9      .1       0  5002.5     .07       0  5008.5      .1       0
  5641.5     .16       0  5882.3      .1       0
Bank Sta=4949,5083.4
XS Rating Curve= 0 ,0
Exp/Cntr=0.3,0.1

Type RM Length L Ch R = 1 ,18801   ,366,366,366
BEGIN DESCRIPTION:
LEFT BEAR CREEK 37.0
END DESCRIPTION:
XS GIS Cut Line= 2
      2746179.51     10018335.89      2747450.38       10019263.
#Sta/Elev= 30
  4314.9 1853.38  4355.3    1852  4384.6 1852.89    4441 1849.54  4499.3 1849.98
  4562.3 1846.37  4627.2    1846    4685 1842.42  4777.8 1840.36  4834.2 1833.31
  4884.4 1829.39  4957.3 1828.31    4964 1824.67  4981.8 1815.43  4984.6 1814.93
  4987.8 1815.43  5085.3 1819.17  5106.1 1822.86  5164.8 1824.06  5242.1 1823.79
  5442.9 1830.08  5478.4 1833.51  5537.1 1843.46  5650.4 1848.97  5708.6 1856.26
  5757.3 1856.54  5786.6 1856.19  5831.1 1857.71    5886 1860.51    5888 1860.51
#Mann= 6 ,-1 , 0
  4314.9      .1       0  4981.8     .07       0  4987.8      .1       0
  5757.3     .16       0  5831.1      .1       0    5886     .16       0
Bank Sta=4964,5164.8
XS Rating Curve= 0 ,0
Exp/Cntr=0.3,0.1

Type RM Length L Ch R = 1 ,18435   ,509,509,509
BEGIN DESCRIPTION:
LEFT BEAR CREEK 36.0
END DESCRIPTION:
XS GIS Cut Line= 2
      2746059.71     10018754.29      2747224.95     10019466.96
#Sta/Elev= 30
  4467.1 1842.41  4510.3  1839.9  4605.1 1837.75  4626.4 1833.55    4669 1828.83
  4690.3 1830.04  4711.8 1827.36  4843.2 1825.07  4932.1 1824.78  4953.4 1825.94
  4959.3 1825.35  4968.9 1822.34  4981.4  1815.3    4993 1814.99  4995.8 1814.49
    4999 1814.99  5026.9 1817.31  5090.8 1817.45  5112.1 1820.43  5136.4 1820.61
    5200 1821.38  5286.3 1822.51  5381.1 1824.04    5462 1827.82  5485.5  1830.9
    5534 1840.28  5594.2 1845.43  5732.9 1851.52  5766.8 1855.09    5833 1854.13
#Mann= 7 ,-1 , 0
  4467.1      .1       0    4993     .07       0    4999      .1       0
  5136.4     .05       0    5200      .1       0  5594.2     .05       0
  5732.9      .1       0
Bank Sta=4968.9,5286.3
XS Rating Curve= 0 ,0
Exp/Cntr=0.3,0.1

Type RM Length L Ch R = 1 ,17926   ,409,409,409
BEGIN DESCRIPTION:
LEFT BEAR CREEK 35.0
END DESCRIPTION:
XS GIS Cut Line= 3
      2745830.59     10019056.41      2746059.74      10019374.1
      2746985.13       10019816.
#Sta/Elev= 30
  4333.8 1836.34    4388 1833.56    4480 1832.99  4579.8 1826.73  4746.3 1823.67
  4806.5 1824.38  4868.2 1820.39  4930.4  1820.4  4948.2 1820.73  4960.8  1817.7
    4985 1811.81  4987.8 1811.31    4991 1811.81  5078.7 1815.42  5084.3 1817.68
  5100.9 1819.88  5108.9 1819.99  5167.4  1818.6  5271.3 1819.31  5458.3 1823.85
  5503.7 1826.78  5543.5 1832.34  5549.1 1831.76  5594.4  1839.3  5617.1 1840.82
  5645.4 1840.09  5662.5 1846.45  5685.2 1851.85  5721.4 1853.38    5751  1852.3
#Mann= 7 ,-1 , 0
  4333.8      .1       0  4579.8     .05       0  4930.4      .1       0
  4960.8     .16       0    4985     .07       0    4991     .16       0
  5108.9      .1       0
Bank Sta=4948.2,5100.9
XS Rating Curve= 0 ,0
Exp/Cntr=0.3,0.1

Type RM Length L Ch R = 1 ,17517   ,464,464,464
BEGIN DESCRIPTION:
LEFT BEAR CREEK 34.0
END DESCRIPTION:
XS GIS Cut Line= 3
      2745715.97     10019092.81       2745976.4     10019743.89
      2746877.48     10020332.46
#Sta/Elev= 30
  4061.1 1837.37  4344.3 1826.58  4350.1 1826.37  4540.2 1823.66  4642.5 1825.59
  4750.2 1818.58  4849.4 1817.61  4908.1 1819.66  4921.8 1818.03  4936.9 1813.33
  4991.2  1808.6  4993.9  1808.1  4997.2  1808.6  5030.4 1809.86  5051.5 1815.09
  5075.3 1817.44  5169.2 1818.46  5226.4 1820.53  5464.8 1826.69  5588.5 1832.15
  5615.6 1838.17  5645.8 1840.52  5651.8 1844.53  5703.1 1864.27  5709.1 1868.67
  5718.2 1871.58  5724.2 1876.52  5750.6 1883.96  5766.5 1886.01  5838.6 1896.87
#Mann= 8 ,-1 , 0
  4061.1      .1       0  4344.3     .05       0  4350.1      .1       0
  4991.2     .07       0  4997.2      .1       0  5226.4     .05       0
  5750.6      .1       0  5766.5     .16       0
Bank Sta=4921.8,5169.2
XS Rating Curve= 0 ,0
Exp/Cntr=0.3,0.1

Type RM Length L Ch R = 1 ,17053   ,367,367,367
BEGIN DESCRIPTION:
LEFT BEAR CREEK 33.0
END DESCRIPTION:
XS GIS Cut Line= 2
      2745585.77     10019243.86      2746012.87     10020634.55
#Sta/Elev= 30
  4001.2 1835.85  4314.9 1822.91    4365  1818.7    4430 1818.48  4492.7 1815.85
    4566 1816.08  4597.3  1817.4    4702 1816.11  4827.5 1817.32  4900.7  1815.9
  4932.1 1817.13  4945.1 1816.01    4953 1813.79  4973.9 1811.23  4980.2 1808.96
  4991.9  1808.4  4994.6  1807.9  4997.9  1808.4  5026.2 1809.71  5050.8 1813.29
  5057.6 1815.77  5068.1 1817.42  5141.3 1823.37  5172.7 1829.93    5187 1834.44
  5258.3 1846.57  5298.2 1849.33  5323.1  1849.5  5402.8 1854.25    5456 1855.95
#Mann= 5 ,-1 , 0
  4001.2      .1       0  4945.1     .16       0  4991.9     .07       0
  4997.9     .16       0  5258.3      .1       0
Bank Sta=4932.1,5068.1
XS Rating Curve= 0 ,0
Exp/Cntr=0.3,0.1

Type RM Length L Ch R = 1 ,16686   ,543,543,543
BEGIN DESCRIPTION:
LEFT BEAR CREEK 32.0
END DESCRIPTION:
XS GIS Cut Line= 4
      2745257.66     10019368.91      2745549.32     10019931.39
      2745455.57     10020728.27       2745679.5     10020988.65
#Sta/Elev= 30
    4098 1838.09  4159.1 1835.57  4204.8 1834.48    4237 1829.19  4264.7 1827.78
  4281.2 1823.21  4286.8 1824.51  4303.3 1821.15    4340 1824.95  4369.7 1818.39
  4430.1 1815.66  4576.5 1814.11  4794.4 1815.28  4868.6 1813.75  4925.3 1816.25
 4940.91 1813.08  4951.7  1809.1  4972.6 1808.51  4975.4 1808.01  4978.6 1808.51
  5056.2 1808.71 5076.14 1813.08  5086.4 1816.75  5106.5 1819.68  5170.3 1819.57
  5327.6 1823.71  5426.2 1828.02  5524.7 1829.53  5601.7 1834.29  5877.4 1846.83
#Mann= 9 ,-1 , 0
    4098     .05       0  4159.1      .1       0  4972.6     .07       0
  4978.6      .1       0  5170.3     .05       0  5327.6      .1       0
  5426.2     .16       0  5524.7      .1       0  5601.7     .16       0
Bank Sta=4940.91,5076.14
XS Rating Curve= 0 ,0
Exp/Cntr=0.3,0.1

Type RM Length L Ch R = 1 ,16143   ,311,311,311
BEGIN DESCRIPTION:
LEFT BEAR CREEK 31.0
END DESCRIPTION:
XS GIS Cut Line= 3
      2745023.28     10019254.35      2745007.65     10020488.68
      2745189.47     10021060.12
#Sta/Elev= 30
  4239.4 1848.31  4282.4 1847.39  4428.8  1840.6  4478.8 1833.47  4508.8 1826.26
  4558.8 1820.79  4828.8  1809.9  4898.8 1811.13  4948.8 1808.41  4995.8 1799.91
  4998.6 1799.41  5001.8 1799.91  5038.8 1802.21  5088.8 1808.86  5158.9  1812.9
    5193 1812.33  5258.9 1812.59  5474.3 1816.99  5500.1 1818.61  5542.1 1817.77
  5615.5 1820.58  5660.3 1819.75    5731 1822.74  5779.1 1822.62  5821.5 1825.07
    5859  1824.5  5940.9 1827.14  5987.9 1826.63  6035.3 1829.05  6073.5 1828.93
#Mann= 7 ,-1 , 0
  4239.4     .05       0  4282.4      .1       0  4995.8     .07       0
  5001.8      .1       0    5193     .05       0  5474.3      .1       0
  5779.1     .05       0
Bank Sta=4948.8,5088.8
XS Rating Curve= 0 ,0
Exp/Cntr=0.3,0.1

Type RM Length L Ch R = 1 ,15832   ,553,553,553
BEGIN DESCRIPTION:
LEFT BEAR CREEK 30.0
END DESCRIPTION:
XS GIS Cut Line= 3
      2744596.19     10019431.38      2744809.74     10020592.85
      2745002.45     10021004.32
#Sta/Elev= 30
    4395 1854.52  4551.4 1847.24  4641.4 1841.77  4656.6 1838.77  4661.8 1835.79
  4695.8 1826.48  4722.8 1815.12  4732.9 1813.28  4833.4 1809.19  4879.7 1809.28
  4946.4 1810.13  4956.6 1809.04  4966.8 1804.96  4971.6  1803.6  4994.3 1798.83
    4997 1798.33  5000.3 1798.83  5043.3 1803.75  5063.2 1803.98  5172.4 1805.67
  5241.3 1812.16  5273.2 1811.37  5325.1 1811.87  5414.2 1813.35  5495.5 1818.19
  5545.6 1818.75  5611.9 1821.19  5674.9 1820.62  5742.6  1823.3  6030.3 1827.16
#Mann= 13 ,-1 , 0
    4395     .05       0  4551.4      .1       0  4695.8     .16       0
  4833.4      .1       0  4879.7     .16       0  4971.6      .1       0
  4994.3     .07       0  5000.3      .1       0  5063.2     .16       0
  5172.4      .1       0  5273.2     .05       0  5325.1      .1       0
  5545.6     .05       0
Bank Sta=4966.8,5172.4
XS Rating Curve= 0 ,0
Exp/Cntr=0.3,0.1

Type RM Length L Ch R = 1 ,15279   ,453,453,453
BEGIN DESCRIPTION:
LEFT BEAR CREEK 29.0
END DESCRIPTION:
XS GIS Cut Line= 4
      2744012.86     10019759.53      2744205.57     10020259.52
      2744742.03     10020691.81      2744877.46     10021014.76
#Sta/Elev= 30
  4240.3 1866.27  4379.9  1851.5  4464.4 1845.88  4489.1 1831.84  4494.4 1835.61
    4502 1830.95  4519.1 1827.56  4543.7 1825.67    4549 1827.94  4566.3 1822.21
    4579 1820.99  4598.3 1823.26  4603.6 1819.39  4628.3 1821.23  4633.6  1818.7
  4652.1 1817.22  4681.8 1811.23  4775.7 1804.51  4916.5 1803.48  4945.3 1801.49
  4966.1 1797.33  4986.9  1797.7  5001.1 1794.91  5009.3 1797.46  5030.1 1796.74
  5063.5 1803.13  5065.3 1803.34  5207.6  1812.4  5428.4 1820.67  5815.3 1827.57
#Mann= 4 ,-1 , 0
  4240.3     .16       0  4681.8      .1       0  4916.5     .09       0
  5063.5      .1       0
Bank Sta=4916.5,5065.3
XS Rating Curve= 0 ,0
Exp/Cntr=0.3,0.1

Type RM Length L Ch R = 1 ,14826   ,287,287,287
BEGIN DESCRIPTION:
LEFT BEAR CREEK 28.0
END DESCRIPTION:
XS GIS Cut Line= 4
      2743585.75     10020332.43      2743919.11     10020400.14
      2744127.44      10020811.6      2744762.82     10021040.75
#Sta/Elev= 30
  4435.6 1931.75  4458.8 1926.56  4509.8 1902.25  4522.4 1894.21  4560.6 1876.42
  4566.8 1871.36  4581.2 1863.85  4611.8 1851.35  4632.3 1839.71  4662.9  1829.1
  4673.2 1823.31  4724.1 1810.82  4754.7    1808  4846.6 1800.65  4891.2 1801.84
  4913.5 1799.08  4963.6 1799.62  5002.3  1791.8  5015.2 1793.29  5047.1 1801.31
  5052.7 1802.47  5091.7 1804.85  5450.7 1802.56  5526.8 1802.26  5613.6 1804.56
  5639.2 1811.47  5644.2 1811.14  5663.3  1816.6  5845.7 1824.15  5912.4 1825.44
#Mann= 9 ,-1 , 0
  4435.6      .1       0  4522.4     .16       0  4560.6      .1       0
  4754.7     .16       0  4891.2     .07       0  5047.1     .16       0
  5450.7      .1       0  5639.2     .16       0  5845.7     .05       0
#XS Ineff= 1 ,-1
    5090 5657.27 1805.63
Permanent Ineff=
       F
Bank Sta=4891.2,5052.7
XS Rating Curve= 0 ,0
Exp/Cntr=0.3,0.1
