HEC-RAS study LIVE OAK CREEK.prj: LIVE OAK CREEK Base Level Engineering

--- LIVE OAK CREEK.g01 (geometry) --- (continued)

Type RM Length L Ch R = 1 ,34232   ,390,390,390
BEGIN DESCRIPTION:
LIVE OAK CREEK 63.0
END DESCRIPTION:
XS GIS Cut Line= 2
      2736608.68      10071666.3      2735293.31     10070899.41
#Sta/Elev= 30
  4388.6 1779.83    4493 1778.08  4614.1 1762.64  4650.9 1759.86  4698.5 1755.79
    4720 1749.47  4725.8 1742.91  4735.7 1740.22  4741.5 1733.15    4763 1721.21
  4784.5 1714.76  4815.4 1711.45  4896.2 1711.85  4960.7 1707.85  4982.2 1702.44
  5000.7 1701.78  5003.4 1701.28  5006.7 1701.78  5056.6 1708.82  5142.6 1708.59
  5174.1 1714.66  5294.1 1721.88  5384.3  1730.8    5542 1733.64  5596.7 1735.99
  5620.8  1741.3  5649.3 1749.73  5714.1 1762.07  5815.8 1770.35  5911.2 1773.92
#Mann= 10 ,-1 , 0
  4388.6      .1       0  4614.1     .16       0  4650.9     .05       0
  4815.4      .1       0  5000.7     .07       0  5006.7      .1       0
  5294.1     .05       0    5542      .1       0  5620.8     .16       0
  5649.3     .05       0
Bank Sta=4784.5,5174.1
XS Rating Curve= 0 ,0
Exp/Cntr=0.3,0.1

Type RM Length L Ch R = 1 ,33842   ,566,566,566
BEGIN DESCRIPTION:
LIVE OAK CREEK 62.0
END DESCRIPTION:
XS GIS Cut Line= 2
      2736953.39      10071282.8      2735401.71     10070681.52
#Sta/Elev= 30
  4246.5 1775.62  4412.6 1774.17  4517.6  1770.4  4619.7 1763.89  4637.9 1752.29
  4644.2 1744.58  4680.8 1717.56  4691.5 1713.28  4712.9 1708.72  4746.3 1708.62
  4959.6 1706.81  4970.3 1704.93  4976.5 1701.55  4998.1 1699.62  5000.8 1699.12
  5004.1 1699.62    5031 1705.11  5060.9 1705.75  5085.5 1713.29  5149.7 1714.93
  5302.8  1719.3  5417.8 1727.55    5622 1737.01  5641.1 1739.95  5678.1 1754.49
  5689.5 1757.01  5710.3 1760.02    5780 1758.92  5867.7 1763.92  5910.6 1766.14
#Mann= 9 ,-1 , 0
  4246.5      .1       0  4517.6     .16       0  4746.3      .1       0
  4998.1     .07       0  5004.1      .1       0  5149.7     .05       0
    5622     .16       0  5689.5     .05       0  5867.7      .1       0
Bank Sta=4691.5,5085.5
XS Rating Curve= 0 ,0
Exp/Cntr=0.3,0.1

Type RM Length L Ch R = 1 ,33276   ,482,482,482
BEGIN DESCRIPTION:
LIVE OAK CREEK 61.0
END DESCRIPTION:
XS GIS Cut Line= 3
      2736953.37     10070957.53       2736361.1      10070404.1
      2735303.15     10070413.81
#Sta/Elev= 30
    4313 1768.07  4382.4 1766.43  4453.7 1768.29  4616.4 1761.54  4721.3 1740.07
  4729.7 1732.88  4736.6 1736.36  4743.9 1728.02  4750.7 1730.63  4764.9 1720.67
  4785.9 1720.68  4793.1 1716.09  4806.8 1713.66  4819.6 1710.93  4856.7 1703.36
  4957.5 1705.48  4995.4 1699.74  4998.2 1699.24  5001.4 1699.74  5040.9  1706.2
  5104.4 1705.59  5136.2 1710.28  5176.2 1717.53  5306.2 1727.47  5645.6 1729.47
  5756.3 1735.63  5843.1 1752.92  6040.5 1766.55  6139.3 1766.67  6181.6 1767.04
#Mann= 11 ,-1 , 0
    4313     .05       0  4382.4     .16       0  4793.1      .1       0
  4806.8     .16       0  4957.5     .05       0  4995.4    .035       0
  5001.4     .05       0  5645.6      .1       0  5843.1     .05       0
  6040.5     .16       0  6139.3     .05       0
Bank Sta=4819.6,5136.2
XS Rating Curve= 0 ,0
Exp/Cntr=0.3,0.1

Type RM Length L Ch R = 1 ,32794   ,689,689,689
BEGIN DESCRIPTION:
LIVE OAK CREEK 60.0
END DESCRIPTION:
XS GIS Cut Line= 2
      2737346.61     10070175.93      2735712.03     10069904.31
#Sta/Elev= 30
  4296.8 1763.53    4447 1761.96  4650.4 1754.83  4730.8 1751.98    4767 1746.58
  4772.1 1748.47  4822.1 1738.74  4827.9 1735.01    4833 1736.05  4872.7 1716.25
  4903.1 1710.07  4929.6 1708.05    4964 1705.55  4974.1  1703.8  4981.7 1699.03
  4991.4 1696.34  4994.1 1695.84  4997.4 1696.34  5015.8 1698.04  5034.9  1704.5
  5065.3 1704.96  5146.4 1703.76  5207.3 1699.45  5247.8 1709.34  5298.5 1728.35
  5572.2 1724.99  5734.4 1728.17  5795.2 1732.08  5863.5 1751.34  5953.8 1754.42
#Mann= 6 ,-1 , 0
  4296.8      .1       0  4650.4     .16       0  4929.6      .1       0
  4981.7     .05       0  4991.4    .035       0  4997.4     .05       0
Bank Sta=4903.1,5247.8
XS Rating Curve= 0 ,0
Exp/Cntr=0.3,0.1

Type RM Length L Ch R = 1 ,32105   ,434,434,434
BEGIN DESCRIPTION:
LIVE OAK CREEK 59.0
END DESCRIPTION:
XS GIS Cut Line= 3
       2737642.7     10070107.94      2736827.15     10069413.75
      2736061.74     10069171.54
#Sta/Elev= 30
    3864 1759.69  4122.7 1761.69  4302.9 1759.53  4418.1 1755.49    4480 1754.29
  4565.6 1749.19  4650.3 1728.08  4707.4 1722.52  4756.8 1714.17  4832.2 1708.75
  4841.3  1707.7  4965.1 1701.23  4993.5 1693.87  4996.3 1693.37  4999.5 1693.87
    5007 1694.76  5020.3 1701.28  5038.5 1701.21  5052.6  1697.3  5090.9 1697.25
  5143.4 1706.77  5154.8 1711.26  5246.5 1713.13  5468.1 1721.31  5510.2  1728.7
  5547.7 1744.21  5562.9 1748.11  5625.9 1759.58  5649.9 1761.33  5737.8 1756.32
#Mann= 8 ,-1 , 0
    3864     .05       0  4122.7      .1       0  4418.1     .16       0
  4832.2      .1       0  4993.5     .07       0  4999.5      .1       0
  5246.5     .05       0  5468.1      .1       0
Bank Sta=4841.3,5143.4
XS Rating Curve= 0 ,0
Exp/Cntr=0.3,0.1

Type RM Length L Ch R = 1 ,31671   ,462,462,462
BEGIN DESCRIPTION:
LIVE OAK CREEK 58.0
END DESCRIPTION:
XS GIS Cut Line= 3
      2737522.17     10069811.09      2737506.55     10069040.22
       2736225.3     10068936.05
#Sta/Elev= 30
  3648.6 1756.98  3878.7 1751.45    4046 1749.73  4079.7 1747.94  4126.1 1739.28
  4156.1 1735.28  4266.1 1727.74  4346.1  1717.8  4396.1 1714.36  4478.1 1711.75
    4687 1710.44  4788.9 1710.34  4864.1 1705.63  4869.2 1705.34  4959.5 1699.88
  4986.6    1693  4989.3  1692.5  4992.6    1693  5039.7 1697.35  5079.9 1697.04
    5149 1702.29  5160.1 1705.38  5170.2 1707.09  5380.9 1713.83  5531.4 1721.77
  5581.5  1730.7  5611.6 1740.99  5631.7 1746.36  5669.4 1753.19  5705.1 1756.55
#Mann= 8 ,-1 , 0
  3648.6      .1       0  3878.7     .05       0  4478.1      .1       0
    4687     .05       0  4864.1      .1       0  4986.6     .07       0
  4992.6      .1       0    5149     .05       0
Bank Sta=4869.2,5160.1
XS Rating Curve= 0 ,0
Exp/Cntr=0.3,0.1

Type RM Length L Ch R = 1 ,31209   ,190,190,190
BEGIN DESCRIPTION:
LIVE OAK CREEK 57.0
END DESCRIPTION:
XS GIS Cut Line= 4
      2738262.64     10068223.98      2737781.82     10068290.56
       2736797.9     10068630.86      2736253.05     10068818.61
#Sta/Elev= 30
  3713.9 1729.62  3889.5 1722.76  3966.4 1721.31  3971.4 1723.03  3990.7 1722.82
  4091.6 1713.76  4172.4 1710.89  4276.9 1703.15  4308.7  1698.4  4351.5 1705.65
  4683.8 1703.76  4839.6 1700.11  4865.5 1696.66  4943.5 1697.27    4959 1696.34
  4975.3 1692.37    5004 1691.15  5006.8 1690.65    5010 1691.15  5021.3 1691.46
  5038.8 1696.86  5083.7 1699.57  5102.3 1704.52  5234.2 1709.32  5291.3 1713.52
  5515.1 1718.23  5603.5 1723.04  5715.8 1734.28  5785.5 1749.47  5816.7  1752.8
#Mann= 3 ,-1 , 0
  3713.9     .05       0    5004     .04       0    5010     .05       0
#XS Ineff= 2 , 0
         4406.25 1706.21
Permanent Ineff=
       T       T
Bank Sta=4683.8,5102.3
XS Rating Curve= 0 ,0
Exp/Cntr=0.3,0.1

Type RM Length L Ch R = 1 ,31019   ,443,443,443
BEGIN DESCRIPTION:
LIVE OAK CREEK 56.0
END DESCRIPTION:
XS GIS Cut Line= 4
      2738273.78     10068101.91      2737785.52     10068157.39
      2737042.16     10068402.35      2736266.97     10068618.34
#Sta/Elev= 30
  3792.1 1726.13  3968.5 1723.05  4149.7 1724.43  4230.2 1719.68  4270.5 1711.15
  4450.8 1703.85  4477.3 1695.85  4509.1 1704.04  4554.2 1705.45  4730.3 1699.85
  4832.1 1701.74    4870 1694.44  4927.4 1694.99  4972.3 1689.93  4975.1 1689.43
  4978.3 1689.93  5132.3 1700.86  5201.6 1703.01  5236.5  1704.4  5313.7 1709.35
  5347.9 1715.94    5409    1718  5553.5 1720.62    5641 1723.16  5661.7 1728.58
  5686.9 1729.43  5703.3 1735.07  5823.7 1741.12  5870.6  1744.4  5870.9  1744.4
#Mann= 10 ,-1 , 0
  3792.1     .05       0  4730.3      .1       0  4972.3     .07       0
  4978.3      .1       0  5201.6     .05       0  5236.5     .08       0
    5409     .05       0  5553.5     .08       0  5823.7     .05       0
  5870.6     .08       0
#XS Ineff= 2 , 0
          4555.4 1705.49
Permanent Ineff=
       T       T
Bank Sta=4832.1,5132.3
XS Rating Curve= 0 ,0
Exp/Cntr=0.3,0.1

Type RM Length L Ch R = 1 ,30576   ,881,881,881
BEGIN DESCRIPTION:
LIVE OAK CREEK 55.0
END DESCRIPTION:
XS GIS Cut Line= 3
      2738220.12     10067982.93      2737360.71     10068014.18
      2736423.34     10067764.21
#Sta/Elev= 30
  4106.1 1724.73  4237.8 1722.05    4381 1723.65    4478 1720.19  4618.1 1702.89
  4648.1 1701.25  4668.1 1697.71  4678.1 1694.22  4688.1 1693.75  4708.1 1700.19
  4718.2 1701.56  4738.2 1701.34  4814.7 1696.18  4855.5 1697.58  4878.3 1697.85
  4898.3 1695.28  4948.3 1695.69  4958.3 1694.25  4964.7 1691.61  4996.4 1689.33
  4999.2 1688.83  5002.4 1689.33  5020.1 1689.48  5065.8 1701.97  5071.9 1704.76
  5082.2 1706.41  5228.6 1714.77  5286.4 1716.17    5579 1718.25  5936.2 1722.56
#Mann= 7 ,-1 , 0
  4106.1      .1       0    4381     .05       0  4855.5      .1       0
  4996.4     .07       0  5002.4      .1       0  5228.6     .05       0
  5286.4      .1       0
Bank Sta=4618.1,5065.8
XS Rating Curve= 0 ,0
Exp/Cntr=0.3,0.1

Type RM Length L Ch R = 1 ,29695   ,550,550,550
BEGIN DESCRIPTION:
LIVE OAK CREEK 54.0
END DESCRIPTION:
XS GIS Cut Line= 2
      2738186.46     10067204.89      2736352.45     10067316.49
#Sta/Elev= 30
  4451.9 1721.47  4515.1 1716.75  4610.2 1712.95  4730.4 1712.73  4850.6 1714.96
  4860.6 1713.88  4880.7  1703.5  4890.7 1700.21  4910.7 1694.13  4940.8 1687.39
  4997.9 1684.75  5000.7 1684.25  5003.9 1684.75  5006.1 1685.84  5012.5 1686.76
    5031 1693.55    5041 1694.77  5131.1 1693.79  5181.2 1696.11  5201.3 1700.18
  5231.3 1701.04  5421.7 1706.78  5511.8 1706.65  5592.3  1709.4  5762.3 1714.22
  6052.8 1717.27  6164.8 1719.86  6253.2 1725.04  6284.6 1729.24  6289.3 1728.58
#Mann= 6 ,-1 , 0
  4451.9      .1       0  4997.9     .07       0  5003.9      .1       0
  5006.1     .05       0  5592.3      .1       0  6284.6     .16       0
Bank Sta=4890.7,5231.3
XS Rating Curve= 0 ,0
Exp/Cntr=0.3,0.1

Type RM Length L Ch R = 1 ,29145   ,695,695,695
BEGIN DESCRIPTION:
LIVE OAK CREEK 53.0
END DESCRIPTION:
XS GIS Cut Line= 3
      2737890.33     10066801.96      2737628.17      10066690.3
      2736411.56     10066952.04
#Sta/Elev= 30
  4592.4 1712.25  4676.6  1713.1  4767.7 1711.29  4774.4  1711.4  4834.7 1706.79
  4852.8 1703.28  4858.3 1703.86  4879.8 1700.49  4915.1 1693.95  4958.9 1690.71
  4969.6 1688.91  4979.3 1685.02  5005.7 1682.82  5008.5 1682.32  5011.7 1682.82
  5030.5 1688.01  5046.6 1690.07    5143 1692.92  5193.4 1696.97  5224.8 1700.23
  5245.2 1703.26  5299.7  1703.8  5388.1 1708.62  5521.5 1712.58  5623.8 1711.78
  5803.7  1713.3    5946 1716.21  6014.3  1720.1  6043.1 1722.94  6121.8 1726.81
#Mann= 9 ,-1 , 0
  4592.4      .1       0  4767.7     .05       0  4774.4      .1       0
  5005.7     .07       0  5011.7      .1       0  5046.6     .05       0
  5193.4      .1       0  5803.7     .05       0    5946      .1       0
Bank Sta=4879.8,5224.8
XS Rating Curve= 0 ,0
Exp/Cntr=0.3,0.1

Type RM Length L Ch R = 1 ,28450   ,589,589,589
BEGIN DESCRIPTION:
LIVE OAK CREEK 52.0
END DESCRIPTION:
XS GIS Cut Line= 2
      2737997.13     10066583.51      2736823.33     10065598.87
#Sta/Elev= 30
  4217.5 1710.68  4301.7 1711.31  4462.5 1702.98  4634.7 1699.18  4736.9  1693.9
  4790.8 1691.31  4933.6 1690.04  5001.2 1679.42  5003.9 1678.92  5007.2 1679.42
    5012 1679.58  5039.3 1692.62  5053.6 1697.12  5067.9 1698.41  5075.7 1697.02
  5082.2 1699.26    5090  1698.4  5096.5 1700.92  5103.3 1699.66  5110.9 1706.19
  5117.4 1706.78  5125.2 1716.15  5131.7 1716.73  5139.5 1721.98  5181.6 1728.11
  5458.2 1738.17  5482.4 1739.08  5606.7 1740.85  5698.6 1739.85  5749.6 1738.29
#Mann= 9 ,-1 , 0
  4217.5      .1       0  4462.5     .05       0  4736.9     .16       0
  5001.2     .07       0  5007.2     .16       0  5458.2      .1       0
  5482.4     .05       0  5606.7      .1       0  5698.6     .05       0
Bank Sta=4634.7,5082.2
XS Rating Curve= 0 ,0
Exp/Cntr=0.3,0.1

Type RM Length L Ch R = 1 ,27861   ,565,565,565
BEGIN DESCRIPTION:
LIVE OAK CREEK 51.0
END DESCRIPTION:
XS GIS Cut Line= 3
      2738186.44     10066369.88        2737667.     10065510.62
      2737346.63     10065437.81
#Sta/Elev= 30
    4092 1710.38  4153.7 1709.94  4239.4 1703.08  4362.1 1698.48  4498.8 1698.63
  4625.3 1699.01  4706.8 1696.24  4809.5 1691.98  4849.1 1687.25  4947.3  1688.8
  4962.8 1687.55  4984.2 1680.42  4995.9 1678.65  4998.7 1678.15  5001.9 1678.65
    5021 1681.67    5034 1686.77  5042.4  1687.1  5057.4 1690.02 5067.27 1696.37
  5079.2 1703.86  5091.3 1716.28  5096.1 1716.28  5102.1 1720.38  5107.3 1726.84
  5115.1  1729.1  5125.3  1728.9  5166.3  1732.9  5217.6 1734.66  5424.6 1735.71
#Mann= 6 ,-1 , 0
    4092      .1       0  4362.1     .05       0  4498.8      .1       0
  4849.1     .16       0  4995.9     .07       0  5001.9     .16       0
Bank Sta=4706.8,5067.27
XS Rating Curve= 0 ,0
Exp/Cntr=0.3,0.1

Type RM Length L Ch R = 1 ,27296   ,680,680,680
BEGIN DESCRIPTION:
LIVE OAK CREEK 50.0
END DESCRIPTION:
XS GIS Cut Line= 3
      2738438.88     10066068.88      2738113.63     10065127.11
      2737741.61     10065040.14
#Sta/Elev= 30
  4153.3 1709.89    4167 1709.62  4183.1 1706.57  4322.9 1694.87    4483 1695.05
    4537 1695.49  4613.7 1696.69  4629.5 1696.13  4634.8 1694.36  4663.6 1687.88
  4686.5 1684.96    4723 1686.71  4772.4 1683.69  4811.3 1688.29    4857 1690.25
    4912 1686.28    4936 1686.61  4990.1  1677.7  4992.9  1677.2  4996.1  1677.7
  5015.7 1679.32  5024.3 1682.85  5029.6 1685.66  5036.9 1695.96  5055.5 1713.69
  5060.8 1716.26    5090 1716.66  5339.8  1726.8  5454.4 1727.68  5531.7 1728.42
#Mann= 10 ,-1 , 0
  4153.3      .1       0  4183.1     .05       0    4483      .1       0
    4537     .05       0  4663.6      .1       0    4912     .16       0
  4990.1     .07       0  4996.1     .16       0    5090      .1       0
  5454.4     .16       0
Bank Sta=4634.8,5036.9
XS Rating Curve= 0 ,0
Exp/Cntr=0.3,0.1

Type RM Length L Ch R = 1 ,26616   ,390,390,390
BEGIN DESCRIPTION:
LIVE OAK CREEK 49.0
END DESCRIPTION:
XS GIS Cut Line= 3
      2738667.64     10066405.27      2738813.26     10065294.97
      2738222.94     10064559.35
#Sta/Elev= 30
  4027.8 1708.82  4251.2 1706.81  4457.5 1702.23  4553.8 1695.44  4584.1 1699.98
  4615.1 1697.77  4692.5  1697.2  4754.5 1694.33  4775.7 1693.44  4846.5 1690.06
  4937.1 1682.96  4967.3 1677.46    4991 1675.97  4993.7 1675.47    4997 1675.97
  5010.1  1677.1  5037.9 1682.51  5057.6 1682.87  5108.5 1683.68  5165.8  1687.4
    5209 1693.37  5229.8 1698.87  5265.1 1702.98  5334.7 1706.23    5429 1706.28
    5631 1704.92  5841.6  1706.1  5948.4 1708.94  6027.2 1713.92  6090.8 1717.41
#Mann= 11 ,-1 , 0
  4027.8      .1       0  4692.5     .05       0  4754.5      .1       0
    4991     .07       0    4997      .1       0  5010.1     .05       0
  5057.6     .16       0  5334.7     .05       0    5429      .1       0
    5631     .16       0  6027.2     .05       0
Bank Sta=4775.7,5209
XS Rating Curve= 0 ,0
Exp/Cntr=0.3,0.1

Type RM Length L Ch R = 1 ,26226   ,564,564,564
BEGIN DESCRIPTION:
LIVE OAK CREEK 48.0
END DESCRIPTION:
XS GIS Cut Line= 3
      2738982.61     10065952.38      2739167.09     10065374.69
       2738628.2     10064850.37
#Sta/Elev= 30
  4295.2 1705.95  4514.2 1703.28  4671.7 1703.63    4690 1704.49  4773.5 1703.98
  4904.2 1703.75  4908.4 1703.39  4915.4 1700.18  4922.6 1698.46 4932.73 1692.28
  4943.7  1686.2  4957.8 1681.53    4972 1675.11  4997.3 1674.01    5000 1673.51
  5003.3 1674.01  5014.4  1676.4  5021.6 1680.54  5028.6 1682.73  5065.4 1683.13
  5099.3 1682.45  5120.6 1684.22  5155.9 1689.12  5247.9 1692.54  5269.1 1694.96
  5290.4 1699.42  5304.1 1701.03  5346.8 1704.63  5628.4 1703.95  5653.5 1703.79
#Mann= 8 ,-1 , 0
  4295.2      .1       0  4671.7     .05       0  4773.5      .1       0
  4997.3     .07       0  5003.3      .1       0  5065.4     .16       0
  5304.1     .05       0  5628.4      .1       0
Bank Sta=4932.73,5247.9
XS Rating Curve= 0 ,0
Exp/Cntr=0.3,0.1

Type RM Length L Ch R = 1 ,25662   ,532,532,532
BEGIN DESCRIPTION:
LIVE OAK CREEK 47.0
END DESCRIPTION:
XS GIS Cut Line= 3
      2740104.01     10065083.41      2739453.51     10064855.25
       2738542.1     10064763.14
#Sta/Elev= 30
  4221.3 1734.56  4298.1 1734.32  4507.7 1731.84  4538.7 1729.27  4545.1 1727.24
  4576.9 1722.44  4638.2 1718.25  4693.7 1713.57  4776.1 1704.26  4812.4 1701.61
  4838.1 1695.95  4882.2 1691.63  4894.8 1690.19  4900.1 1688.72  4910.7 1688.28
  4915.7 1686.42  4955.9 1679.67  4973.2 1673.19  5003.2 1672.13  5005.9 1671.63
  5009.2 1672.13  5036.3 1680.22  5056.4 1680.41  5073.2 1683.38    5231 1690.22
  5378.2 1701.14  5418.3 1702.37    5718 1703.01  5789.1 1703.73  5826.7  1704.1
#Mann= 9 ,-1 , 0
  4221.3     .05       0  4298.1      .1       0  4638.2     .16       0
  4882.2      .1       0  5003.2     .07       0  5009.2      .1       0
    5231     .05       0    5718      .1       0  5789.1     .16       0
Bank Sta=4894.8,5231
XS Rating Curve= 0 ,0
Exp/Cntr=0.3,0.1

Type RM Length L Ch R = 1 ,25130   ,512,512,512
BEGIN DESCRIPTION:
LIVE OAK CREEK 46.0
END DESCRIPTION:
XS GIS Cut Line= 3
      2739918.46     10064553.73      2739568.47     10064353.73
      2739068.48     10064353.73
#Sta/Elev= 30
  4582.2  1728.3  4639.8 1725.09  4708.2 1722.71  4729.8 1720.62  4766.5 1712.89
    4773  1710.2    4801 1702.02  4837.7 1694.07  4853.6 1689.56  4869.4 1687.93
  4896.8  1684.3  4905.4 1681.81  4912.6 1680.34  4962.3 1678.51  4977.4 1676.85
  4982.4 1673.84  4987.8 1673.84  4992.3 1671.08  4995.1 1670.58  4998.3 1671.08
  5015.3  1675.7  5025.3 1676.31  5035.3 1678.88  5095.3 1681.18  5185.3 1688.86
  5205.3 1691.32  5255.3 1693.36  5275.3 1691.94  5365.3 1693.81  5485.3  1699.9
#Mann= 4 ,-1 , 0
  4582.2     .16       0  4905.4      .1       0  4992.3     .07       0
  4998.3      .1       0
Bank Sta=4869.4,5185.3
XS Rating Curve= 0 ,0
Exp/Cntr=0.3,0.1

Type RM Length L Ch R = 1 ,24618   ,536,536,536
BEGIN DESCRIPTION:
LIVE OAK CREEK 45.0
END DESCRIPTION:
XS GIS Cut Line= 3
      2740456.41     10063916.17      2739268.87     10063843.25
      2738586.59     10064322.41
#Sta/Elev= 30
  4239.2 1732.71  4314.4  1732.5  4440.6 1724.98    4678 1709.31  4725.3 1703.93
  4851.6 1690.36  4878.3 1685.98  4928.4 1675.76  4949.3 1675.99  4958.5 1676.08
  4978.5 1671.76  4995.6 1670.46  4998.3 1669.96  5001.6 1670.46  5018.6 1671.29
  5038.6 1677.19  5048.7 1678.49    5143 1684.09  5168.9 1685.79  5229.3 1688.51
  5369.3 1690.98    5559 1691.94  5759.4 1699.29  5843.7 1700.17  5980.6 1700.21
  6118.5  1701.5  6204.8 1705.14  6240.5 1707.55  6255.3 1710.52  6262.7 1709.93
#Mann= 11 ,-1 , 0
  4239.2      .1       0  4314.4     .05       0  4440.6      .1       0
  4725.3     .16       0  4949.3      .1       0  4995.6     .07       0
  5001.6      .1       0    5143     .05       0  5229.3      .1       0
  5843.7     .16       0  5980.6      .1       0
Bank Sta=4878.3,5168.9
XS Rating Curve= 0 ,0
Exp/Cntr=0.3,0.1

Type RM Length L Ch R = 1 ,24082   ,490,490,490
BEGIN DESCRIPTION:
LIVE OAK CREEK 44.0
END DESCRIPTION:
XS GIS Cut Line= 2
       2740404.3     10063384.91      2738737.59     10063327.62
#Sta/Elev= 30
  4360.3  1730.6  4396.2 1730.81  4426.8 1729.04  4540.8 1725.47  4577.4 1722.67
  4706.3 1712.84  4746.4 1706.86  4826.4 1696.59  4831.4  1697.8  4836.4 1696.02
  4869.2 1691.89  4916.5 1684.45  4967.8  1675.1  4993.5 1667.17  4996.3 1666.67
  4999.5 1667.17  5016.5 1668.85  5046.5 1676.35  5066.6 1675.89  5116.6 1679.98
  5206.6 1683.81  5263.6 1684.98  5362.2 1685.46  5490.3 1688.15  5509.1 1688.46
  5616.9 1688.32  5756.5 1693.58    5827 1696.53  5953.7 1695.77    6028 1696.07
#Mann= 14 ,-1 , 0
  4360.3      .1       0  4426.8     .05       0  4577.4      .1       0
  4746.4     .16       0  4869.2      .1       0  4967.8     .05       0
  4993.5    .035       0  4999.5     .05       0  5263.6      .1       0
  5362.2     .05       0  5490.3     .16       0  5509.1     .05       0
  5756.5      .1       0  5953.7     .05       0
Bank Sta=4916.5,5206.6
XS Rating Curve= 0 ,0
Exp/Cntr=0.3,0.1

Type RM Length L Ch R = 1 ,23592   ,508,508,508
BEGIN DESCRIPTION:
LIVE OAK CREEK 43.0
END DESCRIPTION:
XS GIS Cut Line= 2
      2740211.57     10062848.46      2738638.66     10062942.21
#Sta/Elev= 30
  4488.4 1728.77  4541.6 1729.34  4683.9 1720.29    4762 1713.74  4802.1 1707.51
  4822.1 1702.74  4828.1 1699.73  4833.2 1702.31  4842.1 1699.77  4862.2 1698.44
  4892.2 1690.78  4922.3 1691.25  4942.3 1683.78  4963.1 1675.82  4992.3 1666.99
  4999.4 1666.64  5002.2 1666.14  5005.4 1666.64  5012.4 1666.96  5042.5 1675.44
  5072.5 1674.74  5132.6 1679.21  5166.5 1678.31  5242.8 1682.94  5330.7 1684.48
  5483.3 1682.63  5593.5  1684.3  5763.8 1696.24  5915.3 1694.58  6064.1  1694.6
#Mann= 6 ,-1 , 0
  4488.4     .05       0  4683.9     .16       0  4963.1     .05       0
  4999.4    .035       0  5005.4     .05       0  5915.3      .1       0
Bank Sta=4942.3,5242.8
XS Rating Curve= 0 ,0
Exp/Cntr=0.3,0.1

Type RM Length L Ch R = 1 ,23084   ,705,705,705
BEGIN DESCRIPTION:
LIVE OAK CREEK 42.0
END DESCRIPTION:
XS GIS Cut Line= 4
      2739987.62     10062577.62      2739565.75     10062405.75
       2739227.2     10062447.41      2736675.08     10061754.69
#Sta/Elev= 30
  4482.4 1721.19  4622.2 1706.25  4701.5 1697.43  4913.4 1681.66  4955.3  1677.9
  4975.5 1668.19  5002.7 1665.92  5005.5 1665.42  5008.7 1665.92  5047.6 1673.68
  5159.5 1675.43  5165.6 1675.96  5308.7 1681.32  5347.7 1681.71    5516 1683.67
  5635.1 1692.17  5694.7 1694.49    5766 1697.56  5867.1 1700.47  6586.3 1725.27
  6843.4 1731.57  7146.3 1748.57  7262.1 1759.75  7409.4  1773.4  7528.9 1771.14
  7600.6 1777.85    7638 1780.93  7757.4  1774.6    7795 1777.93  7923.5 1785.92
#Mann= 16 ,-1 , 0
  4482.4      .1       0  4622.2     .16       0  4701.5      .1       0
  5002.7     .07       0  5008.7      .1       0  5159.5     .16       0
  5165.6      .1       0  5308.7     .05       0  5635.1      .1       0
  5694.7     .05       0    5766      .1       0  5867.1     .05       0
  6586.3     .16       0  7262.1      .1       0  7600.6     .05       0
    7795     .16       0
Bank Sta=4913.4,5347.7
XS Rating Curve= 0 ,0
Exp/Cntr=0.3,0.1

Type RM Length L Ch R = 1 ,22379   ,616,616,616
BEGIN DESCRIPTION:
LIVE OAK CREEK 41.0
END DESCRIPTION:
XS GIS Cut Line= 3
      2740123.06     10062452.64      2739263.66     10061890.12
      2736794.92     10060858.88
#Sta/Elev= 30
  3851.9  1712.2  3963.8 1705.02  4005.9    1699  4299.1 1683.11  4490.8  1680.6
  4531.9 1679.06  4546.4 1678.68  4636.4 1675.77  4910.2 1673.66  4976.1 1669.06
  5000.9 1663.63  5003.6 1663.13  5006.9 1663.63  5063.5 1678.55  5102.7 1680.63
  5164.5 1686.62  5217.6 1685.92  5270.6 1693.77    5329 1694.01  5400.5 1702.09
  5559.6 1709.59  6055.3 1748.43  6664.6 1763.97  6949.3 1768.42  6981.8  1769.4
  7012.1 1772.67  7160.4 1766.84  7329.3 1778.97    7473 1785.91  7554.5 1789.65
#Mann= 14 ,-1 , 0
  3851.9      .1       0  4299.1     .05       0  4531.9      .1       0
  4546.4     .16       0  4636.4      .1       0  4976.1     .05       0
  5000.9     .04       0  5006.9     .05       0  5102.7     .16       0
  6664.6      .1       0  6949.3     .05       0  6981.8     .16       0
  7329.3     .05       0    7473      .1       0
Bank Sta=4490.8,5102.7
XS Rating Curve= 0 ,0
Exp/Cntr=0.3,0.1

Type RM Length L Ch R = 1 ,21763   ,478,478,478
BEGIN DESCRIPTION:
LIVE OAK CREEK 40.0
END DESCRIPTION:
XS GIS Cut Line= 3
      2740185.56     10062270.36      2739591.79     10061535.96
      2739414.71     10060879.74
#Sta/Elev= 30
  3946.3 1697.17  4027.4 1692.68    4184 1690.63  4276.3 1683.05  4347.2 1679.19
  4566.3 1681.86  4674.9 1680.21  4687.8 1679.28  4724.5 1672.22  4831.8  1673.9
  4944.8 1670.71  4965.9 1668.14  4999.5 1661.55  5003.9 1661.09  5006.7 1660.59
  5009.9 1661.09  5017.3  1662.5  5027.7 1666.79  5035.3 1671.87  5058.7 1680.21
  5075.2 1685.55  5080.4 1684.85  5100.2 1688.02  5214.1 1688.42  5253.2 1690.47
    5297 1694.36  5344.2 1702.46    5379 1705.63  5460.2 1706.07  5570.4 1710.77
#Mann= 8 ,-1 , 0
  3946.3     .05       0  4566.3     .16       0  4831.8      .1       0
  4999.5     .16       0  5003.9     .07       0  5009.9     .16       0
  5253.2     .05       0  5460.2      .1       0
Bank Sta=4674.9,5058.7
XS Rating Curve= 0 ,0
Exp/Cntr=0.3,0.1

Type RM Length L Ch R = 1 ,21285   ,472,472,472
BEGIN DESCRIPTION:
LIVE OAK CREEK 39.0
END DESCRIPTION:
XS GIS Cut Line= 3
      2740357.41     10062223.45      2739945.95     10061103.66
      2740133.46     10060733.87
#Sta/Elev= 30
  3996.8  1694.5  4152.1 1689.82  4297.2 1689.76  4335.1 1689.72  4441.6 1679.92
  4548.1 1676.66  4552.9 1676.69  4667.7 1676.61  4725.2 1679.14  4742.3 1680.12
  4784.9 1678.29  4838.1 1675.72  4867.5 1672.29  4907.2 1668.19  4955.3 1668.35
  4993.3 1660.74  5005.6 1660.44  5008.3 1659.94  5011.6 1660.44  5029.9  1667.1
  5054.3  1671.7  5072.5 1677.61  5079.4 1680.98  5109.9  1689.2  5165.5    1694
  5206.5 1695.15  5231.6 1697.72  5413.9 1696.75  5495.9 1699.79  5604.4 1700.79
#Mann= 11 ,-1 , 0
  3996.8      .1       0  4297.2     .05       0  4335.1      .1       0
  4441.6     .05       0  4548.1      .1       0  4552.9     .05       0
  4725.2      .1       0  4867.5     .16       0  5005.6     .07       0
  5011.6     .16       0  5231.6      .1       0
Bank Sta=4784.9,5072.5
XS Rating Curve= 0 ,0
Exp/Cntr=0.3,0.1

Type RM Length L Ch R = 1 ,20813   ,395,395,395
BEGIN DESCRIPTION:
LIVE OAK CREEK 38.0
END DESCRIPTION:
XS GIS Cut Line= 3
      2740568.48     10061653.78      2740468.47     10061253.73
      2740418.46      10060853.7
#Sta/Elev= 30
  4586.7 1687.46  4608.1 1685.92  4616.7 1685.26    4629 1684.02  4741.4 1673.84
  4769.7 1671.52  4813.2  1672.9  4834.1 1673.16  4862.5 1671.37  4893.4 1668.49
  4898.6 1669.14  4934.6 1666.19  4968.1 1667.22    4981 1665.98  4993.5 1659.87
  4996.2 1659.37  4999.5 1659.87  5036.8 1662.55  5041.9 1661.73  5059.5 1669.06
 5077.05 1674.63  5089.8 1682.62  5109.9 1690.56  5117.5 1692.29  5225.2 1698.77
  5283.8 1701.83  5341.7 1703.34  5351.8 1702.63  5388.5 1704.89  5402.2 1705.38
#Mann= 10 ,-1 , 0
  4586.7      .1       0  4608.1     .05       0  4616.7      .1       0
    4629     .05       0  4813.2      .1       0  4862.5     .16       0
  4993.5     .07       0  4999.5     .16       0  5225.2     .05       0
  5388.5      .1       0
Bank Sta=4741.4,5077.05
XS Rating Curve= 0 ,0
Exp/Cntr=0.3,0.1

Type RM Length L Ch R = 1 ,20418   ,542,542,542
BEGIN DESCRIPTION:
LIVE OAK CREEK 37.0
END DESCRIPTION:
XS GIS Cut Line= 3
       2740784.5     10061869.27      2740883.45     10061119.29
      2740452.33     10060776.47
#Sta/Elev= 30
  4431.6 1688.35  4568.5 1686.87  4653.6 1687.04  4765.8  1678.6  4810.7 1676.44
  4850.7 1672.51  4901.2 1666.21  4962.8 1663.79    4989 1659.31  4991.7 1658.81
    4995 1659.31  5012.1 1659.79  5019.2 1661.62  5031.3 1665.16  5062.6 1667.49
  5082.7 1671.54  5102.9  1677.2  5109.8 1680.97  5114.9 1681.44  5123.1 1684.34
  5133.2 1686.05    5160 1686.52  5366.3 1684.85    5434 1686.05  5475.4 1687.41
  5555.8 1690.37  5623.8 1696.14  5672.3 1696.82  5701.1 1699.74  5738.9 1701.58
#Mann= 11 ,-1 , 0
  4431.6     .05       0  4568.5      .1       0  4765.8     .05       0
    4989    .035       0    4995     .05       0  5019.2     .16       0
    5160      .1       0    5434     .05       0  5475.4      .1       0
  5555.8     .05       0  5623.8      .1       0
Bank Sta=4850.7,5082.7
XS Rating Curve= 0 ,0
Exp/Cntr=0.3,0.1

Type RM Length L Ch R = 1 ,19876   ,581,581,581
BEGIN DESCRIPTION:
LIVE OAK CREEK 36.0
END DESCRIPTION:
XS GIS Cut Line= 3
      2741998.06     10061457.84      2741445.95      10061249.5
      2740555.29     10060770.31
#Sta/Elev= 30
  4325.5 1715.44  4536.3 1706.02  4581.1 1704.48  4632.1 1699.05  4637.5 1699.88
  4662.3 1695.68  4667.6 1696.35  4747.5 1686.97  4788.6 1684.66  4807.9 1682.22
  4827.4 1676.65  4838.1 1671.66  4870.2 1662.82  4934.1 1662.72  4996.8 1658.53
  4999.5 1658.03  5002.8 1658.53    5003 1658.56  5065.5 1663.59  5094.4 1663.94
  5109.3 1667.22  5147.5 1666.85    5197 1671.63  5287.5 1685.13  5541.8 1685.01
  5599.6 1684.22  5700.1 1684.29  5820.7 1688.18  5906.8 1691.75    5927  1692.6
#Mann= 11 ,-1 , 0
  4325.5     .05       0  4536.3      .1       0  4581.1     .05       0
  4788.6     .16       0  4996.8     .07       0  5002.8     .16       0
    5003      .1       0  5541.8     .05       0  5599.6      .1       0
  5820.7     .05       0  5906.8      .1       0
Bank Sta=4838.1,5197
XS Rating Curve= 0 ,0
Exp/Cntr=0.3,0.1

Type RM Length L Ch R = 1 ,19295   ,713,713,713
BEGIN DESCRIPTION:
LIVE OAK CREEK 35.0
END DESCRIPTION:
XS GIS Cut Line= 2
      2742034.48      10060749.5       2740633.5     10060791.16
#Sta/Elev= 30
    4624 1709.68  4710.1 1704.43  4730.1 1701.67  4774.2 1700.67  4800.1 1698.27
  4840.1 1701.37  4920.1 1699.56  4929.9 1695.43  4934.9 1694.62  4940.2 1687.94
  4970.2  1669.5  4980.2 1664.12  4997.2 1657.49  4999.9 1656.99  5003.2 1657.49
  5030.2 1661.31  5133.1 1659.07  5200.3  1663.3  5260.3 1661.56  5273.2 1662.48
  5295.4 1666.46  5310.3  1669.5  5350.3 1678.29  5367.3 1679.68  5466.1 1683.86
  5541.5 1683.01  5691.4 1683.73  5902.3  1683.7  5921.8 1684.31  6025.6 1688.73
#Mann= 12 ,-1 , 0
    4624     .05       0  4774.2     .16       0  4997.2    .035       0
  5003.2     .16       0  5133.1      .1       0  5295.4     .05       0
  5367.3      .1       0  5466.1     .05       0  5541.5      .1       0
  5691.4     .05       0  5902.3      .1       0  5921.8     .05       0
Bank Sta=4970.2,5310.3
XS Rating Curve= 0 ,0
Exp/Cntr=0.3,0.1

Type RM Length L Ch R = 1 ,18582   ,523,523,523
BEGIN DESCRIPTION:
LIVE OAK CREEK 34.0
END DESCRIPTION:
XS GIS Cut Line= 3
      2741815.75      10060374.5      2741326.16     10060155.75
      2740613.02     10060556.57
#Sta/Elev= 30
    4364 1699.92    4528 1694.61  4613.5 1693.64  4689.6 1691.95  4695.9 1689.67
  4701.4 1690.81  4719.2 1688.02  4724.6  1690.6  4742.4 1688.55  4747.8 1690.34
  4765.6 1688.51  4771.1 1689.99  4788.2 1680.95  4794.3 1674.47  4799.7 1677.17
  4802.6 1675.64  4817.5 1668.36  4822.9 1669.75    4832  1666.6  4840.7 1664.78
  4910.6 1658.78  4969.9 1656.75  5004.5 1652.31  5007.2 1651.81  5010.5 1652.31
  5035.2 1660.35  5094.2 1665.85  5191.1 1680.17  5601.7 1682.27  5718.3 1684.46
#Mann= 5 ,-1 , 0
    4364     .05       0  4613.5     .16       0  4802.6     .05       0
  5004.5     .04       0  5010.5     .05       0
Bank Sta=4832,5094.2
XS Rating Curve= 0 ,0
Exp/Cntr=0.3,0.1

Type RM Length L Ch R = 1 ,18059   ,498,498,498
BEGIN DESCRIPTION:
LIVE OAK CREEK 33.0
END DESCRIPTION:
XS GIS Cut Line= 4
      2741690.78      10060233.9      2741138.66     10059707.83
      2740925.12     10059739.08      2740451.15      10060728.7
#Sta/Elev= 30
  4139.4  1693.2  4225.9 1690.68  4261.4 1692.64  4310.8 1688.92  4358.5 1688.74
    4507 1680.67  4664.7 1677.54    4714 1678.88  4735.4 1675.15  4756.5 1677.35
  4770.7 1675.97  4777.9  1672.5  4784.8 1673.23    4799 1664.76 4809.66 1663.83
  4827.3 1660.42    4898 1656.73  4942.8 1657.65  4972.6 1657.39  4983.1 1653.49
  5000.3 1651.67    5003 1651.17  5006.3 1651.67    5074 1664.06  5147.8 1674.33
  5223.1 1677.95  5374.4  1677.3  5929.4 1683.83  6090.5 1690.05  6215.1 1698.94
#Mann= 8 ,-1 , 0
  4139.4     .05       0  4358.5     .16       0    4507     .05       0
  4942.8      .1       0  5000.3     .07       0  5006.3      .1       0
  5223.1     .05       0  6090.5      .1       0
Bank Sta=4809.66,5074
XS Rating Curve= 0 ,0
Exp/Cntr=0.3,0.1

Type RM Length L Ch R = 1 ,17561   ,443,443,443
BEGIN DESCRIPTION:
LIVE OAK CREEK 32.0
END DESCRIPTION:
XS GIS Cut Line= 3
      2741753.25     10060239.08      2741018.87     10059291.16
      2740258.46     10058858.88
#Sta/Elev= 30
  3704.5 1695.32  3862.1 1687.93  4103.4 1680.08    4439  1679.1  4503.1 1675.81
  4524.2 1670.26  4646.1 1662.55  4702.2 1658.04  4760.2 1656.49  4787.3 1652.03
    4810  1652.5  4845.3 1657.36  4887.7 1657.69  4910.8 1655.52  4968.3 1654.22
  4993.1 1651.28  4995.8 1650.78  4999.1 1651.28  5011.5 1652.51 5035.51 1662.02
    5049  1669.9  5151.4  1679.4  5232.1 1698.13  5318.6 1709.96  5334.4 1710.32
  5377.7  1704.9  5415.2 1704.39  5490.1 1714.13  5599.4  1721.7  5778.3 1721.97
#Mann= 7 ,-1 , 0
  3704.5     .05       0    4439      .1       0  4524.2     .05       0
  4910.8     .16       0  4993.1     .07       0  4999.1     .16       0
  5599.4      .1       0
Bank Sta=4646.1,5035.51
XS Rating Curve= 0 ,0
Exp/Cntr=0.3,0.1

Type RM Length L Ch R = 1 ,17118   ,615,615,615
BEGIN DESCRIPTION:
LIVE OAK CREEK 31.0
END DESCRIPTION:
XS GIS Cut Line= 3
      2741820.96     10060207.85      2741367.83     10059160.96
      2740899.09     10058374.51
#Sta/Elev= 30
  3789.1 1695.38  4083.6 1682.72  4392.9 1676.56  4614.9 1676.88  4718.2 1669.31
  4794.8 1665.81    4895 1660.14  4935.4 1653.16  4978.2 1651.97  4990.8 1649.35
  4993.6 1648.85  4996.8 1649.35  5030.8 1652.58    5042 1651.39  5073.6 1655.02
    5095 1654.74  5124.5 1660.31  5137.8 1663.19  5153.4 1669.82  5159.5 1676.73
  5174.8 1684.78  5190.4 1699.78  5196.2 1701.42    5206  1712.1  5217.7 1719.06
  5227.4 1719.81  5408.4 1718.33  5509.7 1713.43    5839 1711.14  5845.4 1711.07
#Mann= 7 ,-1 , 0
  3789.1     .05       0  4718.2      .1       0  4794.8     .05       0
  4990.8    .035       0  4996.8     .05       0    5042     .16       0
    5839      .1       0
Bank Sta=4895,5124.5
XS Rating Curve= 0 ,0
Exp/Cntr=0.3,0.1

Type RM Length L Ch R = 1 ,16503   ,430,430,430
BEGIN DESCRIPTION:
LIVE OAK CREEK 30.0
END DESCRIPTION:
XS GIS Cut Line= 3
      2742024.08     10060129.75        2741972.     10059160.96
      2741529.26     10058681.76
#Sta/Elev= 30
  3954.9 1687.92    4001  1684.4  4051.1 1684.76  4201.3 1679.11  4511.7 1674.75
  4760.1 1673.41  4782.1 1673.24  4822.2 1669.03  4860.2 1661.25  4882.3  1659.2
  4897.5 1655.87  4925.1 1652.67  4947.1 1647.81  4993.4 1646.74  4996.1 1646.24
  4999.4 1646.74  5024.7 1650.26  5045.7 1650.08  5110.4 1653.79  5166.4 1659.32
  5244.2 1667.32  5272.5 1668.97  5279.3 1668.23  5286.7 1669.78  5293.5 1668.81
  5321.9 1669.48  5345.4  1672.2  5399.6 1676.79  5550.6 1685.68  5577.5 1690.24
#Mann= 8 ,-1 , 0
  3954.9     .05       0  4760.1      .1       0  4860.2     .05       0
  4993.4    .035       0  4999.4     .05       0  5110.4     .16       0
  5345.4      .1       0  5550.6     .16       0
Bank Sta=4882.3,5166.4
XS Rating Curve= 0 ,0
Exp/Cntr=0.3,0.1

Type RM Length L Ch R = 1 ,16073   ,769,769,769
BEGIN DESCRIPTION:
LIVE OAK CREEK 29.0
END DESCRIPTION:
XS GIS Cut Line= 3
      2742699.29     10060173.83      2742522.21     10059153.01
      2741504.84     10058462.03
#Sta/Elev= 30
  3743.2 1689.21  3837.8 1684.42  3952.1  1675.3  4066.4  1672.4  4578.6 1672.38
    4677 1674.69  4858.5 1673.77  4904.7 1672.43  4932.1 1665.67    4962 1662.09
    4968 1659.14  4976.9 1655.61    4983 1648.24  4994.9 1644.23  4997.6 1643.73
  5000.9 1644.23  5025.8 1646.02  5069.8 1647.32  5098.8 1650.21  5126.7 1649.71
  5154.3 1653.04  5228.4 1655.69  5255.5 1659.48  5306.3 1669.15  5355.7 1672.91
  5387.1 1675.53  5557.8 1673.23  5715.3 1675.63  5828.9 1680.25  6009.1 1688.74
#Mann= 11 ,-1 , 0
  3743.2      .1       0  4578.6     .05       0  4858.5      .1       0
  4994.9     .07       0  5000.9      .1       0  5025.8     .05       0
  5098.8      .1       0  5154.3     .05       0  5355.7     .16       0
  5715.3      .1       0  5828.9     .16       0
Bank Sta=4968,5255.5
XS Rating Curve= 0 ,0
Exp/Cntr=0.3,0.1

Type RM Length L Ch R = 1 ,15304   ,418,418,418
BEGIN DESCRIPTION:
LIVE OAK CREEK 28.0
END DESCRIPTION:
XS GIS Cut Line= 3
      2743063.88     10059104.37       2743036.1     10058534.95
       2741643.7     10058003.69
#Sta/Elev= 30
  4226.6 1672.89  4347.4 1673.21  4627.7 1670.29  4832.6 1671.47    4867    1672
  4872.3 1671.26  4890.5 1667.53  4902.4 1661.61  4911.9  1658.7  4927.1 1655.96
  4933.3  1653.3  4987.3 1643.53  5003.7 1643.29  5006.4 1642.79  5009.7 1643.29
    5012 1643.36  5018.9 1646.28  5029.6 1647.59  5061.5 1649.11  5091.6  1649.3
  5168.8 1656.21  5225.6 1661.42  5240.9 1662.74  5291.4 1667.34  5376.3 1668.52
  5414.9 1670.95  5532.7 1673.13  5693.2 1672.19  6003.6    1674    6287 1680.67
#Mann= 7 ,-1 , 0
  4226.6     .05       0  4832.6      .1       0  5003.7     .07       0
  5009.7      .1       0  5225.6     .05       0  5240.9      .1       0
  5414.9     .05       0
Bank Sta=4927.1,5168.8
XS Rating Curve= 0 ,0
Exp/Cntr=0.3,0.1

Type RM Length L Ch R = 1 ,14886   ,274,274,274
BEGIN DESCRIPTION:
LIVE OAK CREEK 27.0
END DESCRIPTION:
XS GIS Cut Line= 2
      2743407.67     10058260.67      2742247.92     10057746.77
#Sta/Elev= 30
    4613 1667.73  4719.8 1668.71  4791.6 1668.85  4861.4 1670.27  4884.7 1669.68
  4913.4 1662.58  4929.3 1660.11  4951.2 1653.63  4965.5 1649.93  4972.2  1646.5
  4983.3  1643.2  4994.9 1641.35  5002.9 1641.33  5005.6 1640.83  5008.9 1641.33
    5012 1642.75  5035.3 1647.08  5064.1 1648.32  5126.2 1648.59  5202.8 1654.12
    5204 1654.21  5279.1 1658.63  5337.9 1659.82  5399.6 1663.55  5406.4 1664.95
  5421.5 1666.03  5458.4 1665.57  5518.3 1667.32  5554.4 1668.24  5881.5 1671.44
#Mann= 9 ,-1 , 0
    4613     .05       0  4719.8      .1       0  4972.2     .05       0
  5002.9    .035       0  5008.9     .05       0    5204     .16       0
  5337.9     .05       0  5518.3     .16       0  5554.4     .05       0
Bank Sta=4951.2,5202.8
XS Rating Curve= 0 ,0
Exp/Cntr=0.3,0.1

Type RM Length L Ch R = 1 ,14612   ,507,507,507
BEGIN DESCRIPTION:
LIVE OAK CREEK 26.0
END DESCRIPTION:
XS GIS Cut Line= 2
     2743340.379     10057933.75      2742438.87     10057534.95
#Sta/Elev= 30
  4796.7 1669.12  4862.3 1668.77  4879.9 1669.23  4885.4 1668.82  4903.2 1666.55
    4917 1663.39  4926.5 1660.76  4938.9 1654.39  4949.8 1652.11  4955.3  1650.1
  4971.7  1644.9  4978.6 1641.98  5007.1 1639.91  5015.4 1640.94  5025.2 1643.09
  5030.6 1645.76  5037.3 1646.32  5053.9 1646.99    5106 1646.69  5152.6 1650.43
  5190.4 1652.26  5199.2 1652.74  5321.1  1657.2  5378.6 1657.69  5463.7 1663.18
  5485.6 1662.11  5562.1 1662.87  5697.9 1666.14  5721.2 1667.44  5780.4 1668.42
#Mann= 3 ,-1 , 0
  4796.7     .05       0  4955.3    .035       0  5190.4     .05       0
Bank Sta=4949.8,5199.2
XS Rating Curve= 0 ,0
Exp/Cntr=0.3,0.1

Type RM Length L Ch R = 1 ,14105   ,239,239,239
BEGIN DESCRIPTION:
LIVE OAK CREEK 25.0
END DESCRIPTION:
XS GIS Cut Line= 4
      2744337.54     10058151.65      2743837.53     10057537.05
      2743407.63     10057406.48      2742807.77     10057198.44
#Sta/Elev= 30
  3660.8  1695.6  3766.7 1690.09  3822.5 1687.02  3843.3 1680.76  3857.7 1679.11
  3915.1  1676.8  3964.7 1669.39  4121.3 1659.44  4156.4 1651.97  4185.2 1659.05
    4206 1657.97  4269.9 1662.75  4333.8 1664.68  4348.2 1662.69    4369 1664.45
  4753.5 1664.62  4912.2 1659.11  4943.8  1654.6  4952.8 1650.87    4984    1641
  4996.5 1639.29  5046.3 1645.36  5196.6 1646.64  5227.8  1650.8  5258.9 1651.22
  5295.3 1659.64  5326.5 1670.54  5352.3 1674.67    5508 1685.91  5537.3 1687.52
#Mann= 8 ,-1 , 0
  3660.8     .05       0  3766.7      .1       0  3915.1     .16       0
  3964.7     .08       0  4912.2     .05       0  5258.9     .07       0
  5258.9     .08       0    5508     .05       0
#XS Ineff= 2 , 0
         4748.96  1664.8
Permanent Ineff=
       T       T
Bank Sta=4952.8,5258.9
XS Rating Curve= 0 ,0
Exp/Cntr=0.3,0.1

Type RM Length L Ch R = 1 ,13866   ,178,178,178
XS GIS Cut Line= 5
      2744365.29     10058061.33      2743985.59      10057434.8
      2743795.49     10057257.72      2743477.78     10057156.16
      2742782.97     10057137.94
#Sta/Elev= 30
  3482.3 1693.01  3543.8 1690.18  3559.2 1685.83  3644.6 1682.72  3681.4 1676.03
  3748.4 1671.76  3770.6 1667.84  3776.5 1669.43  3791.9 1665.12  3797.8 1666.79
  3819.1 1662.42  3871.5 1660.93  3877.3 1658.83    3887 1660.52  3892.8 1657.84
  3908.3  1659.9  3958.9 1651.64  4009.1 1659.42  4241.8 1664.06  4468.5 1657.62
  4795.8    1654  4897.6 1648.34  4997.4 1638.53  5067.7 1641.83  5107.7 1649.47
  5147.7 1655.91  5167.7 1662.47  5197.7 1663.68  5237.7 1672.02  5503.3 1688.85
#Mann= 3 , 0 , 0
  3482.3     .16       0  4897.6     .07       0  5107.7     .16       0
#XS Ineff= 2 , 0
         4232.37 1664.26
Permanent Ineff=
       T       T
Bank Sta=4897.6,5107.7
XS Rating Curve= 0 ,0
Exp/Cntr=0.3,0.1

Type RM Length L Ch R = 1 ,13688   ,359,359,359
BEGIN DESCRIPTION:
LIVE OAK CREEK 24.0
END DESCRIPTION:
XS GIS Cut Line= 4
      2744391.83     10057460.84      2743977.07     10057142.59
      2743612.49     10056996.76       2742768.7     10056972.45
#Sta/Elev= 30
  3783.1 1671.07  3798.3 1669.64    3869 1663.19  3933.4 1652.39  3954.2 1651.95
  4132.8 1655.89  4176.3 1660.98  4217.9 1656.72  4261.5 1661.99  4336.7    1664
  4455.7 1653.41  4636.1 1649.31  4671.1 1646.25    4690 1648.75  4695.4    1646
  4732.6 1642.77  4752.6 1644.11  4812.6 1655.36  4892.7 1653.88  4912.7 1649.03
  4942.7 1642.96  4992.5 1638.44  5042.7 1641.52  5082.7 1649.76  5132.8 1665.84
  5162.8 1669.59  5192.8 1667.93  5222.8 1672.87  5342.8 1682.16  5542.7 1685.02
#Mann= 5 ,-1 , 0
  3783.1     .05       0  3798.3     .16       0  4912.7     .05       0
  4912.7     .07       0  5082.7     .16       0
#XS Ineff= 2 ,-1
  3819.5 4331.95 1663.97 4404.56 4815.35 1655.22
Permanent Ineff=
       T       T
Bank Sta=4912.7,5082.7
XS Rating Curve= 0 ,0
Exp/Cntr=0.3,0.1

Type RM Length L Ch R = 1 ,13329   ,492,492,492
XS GIS Cut Line= 4
      2744105.39     10056924.39      2743706.95     10056713.45
      2743222.57      10056617.1       2742925.7     10056653.55
#Sta/Elev= 30
  4299.6 1678.74  4328.7 1677.04    4364 1677.11  4394.7 1675.13  4444.4 1667.07
  4482.7 1662.12  4521.1  1654.5  4533.7 1653.31  4750.4 1647.92  4769.3 1645.78
  4774.5  1644.3  4825.6 1639.34  4850.8 1639.61  4876.7 1641.89  4881.8 1640.36
  4942.6 1642.76  4993.3  1637.7    5014 1639.47  5024.2 1641.74  5035.2    1647
    5065 1659.49  5095.5 1668.04  5105.7 1668.77  5183.4 1667.68  5228.1  1668.7
  5260.6 1670.95  5298.8 1677.41    5319 1678.76  5399.6 1679.68  5543.4 1678.73
#Mann= 3 , 0 , 0
  4299.6     .16       0  4750.4     .07       0  5035.2     .16       0
Bank Sta=4750.4,5035.2
XS Rating Curve= 0 ,0
Exp/Cntr=0.3,0.1

Type RM Length L Ch R = 1 ,12837   ,562,562,562
BEGIN DESCRIPTION:
LIVE OAK CREEK 23.0
END DESCRIPTION:
XS GIS Cut Line= 2
      2744331.34     10056690.84      2743526.25     10056123.87
#Sta/Elev= 30
  4346.1 1677.16  4533.1 1663.47  4590.5 1657.25  4647.1 1653.39  4676.7  1651.9
  4697.7 1652.54  4712.5 1651.44  4718.6 1652.12  4727.3 1651.07  4733.4 1651.54
  4748.2 1649.97  4769.1 1649.64  4783.9 1648.36  4834.4    1647    4891 1644.55
  4935.4 1643.87  4971.1 1642.25  4991.8 1637.26  5048.7 1641.19  5057.4 1643.14
  5071.2  1647.5  5084.4 1649.28  5093.1 1649.12  5107.9 1651.43  5128.8 1658.47
  5143.6 1660.98  5193.5 1661.58    5215 1662.48  5242.5 1667.64  5330.8 1669.55
#Mann= 3 ,-1 , 0
  4346.1     .16       0  4935.4     .07       0  5057.4     .16       0
Bank Sta=4971.1,5057.4
XS Rating Curve= 0 ,0
Exp/Cntr=0.3,0.1

Type RM Length L Ch R = 1 ,12275   ,491,491,491
BEGIN DESCRIPTION:
LIVE OAK CREEK 22.0
END DESCRIPTION:
XS GIS Cut Line= 2
      2744586.54     10056242.95      2743798.41     10055613.57
#Sta/Elev= 30
  4520.9 1676.81  4582.4 1676.43  4619.1 1674.53  4660.7 1669.79  4710.4  1659.8
  4739.2 1656.25  4788.8  1651.8  4860.9 1649.41  4902.5 1644.31  4953.5 1642.34
  4960.1 1641.85  5003.1 1637.04  5073.8 1639.93  5088.2 1642.74  5102.6 1644.59
  5137.9 1652.14  5151.9 1654.17  5158.7 1656.49  5173.1 1658.89  5187.5 1659.79
  5230.7 1658.78  5259.6 1659.22  5358.8 1663.52  5429.3 1668.02  5472.5 1668.37
  5493.3 1669.72  5501.3  1671.5  5522.1 1674.38  5526.3 1676.92  5529.5 1676.92
#Mann= 3 ,-1 , 0
  4520.9     .16       0  4960.1     .07       0  5088.2     .16       0
Bank Sta=4953.5,5088.2
XS Rating Curve= 0 ,0
Exp/Cntr=0.3,0.1

Type RM Length L Ch R = 1 ,11784   ,539,539,539
BEGIN DESCRIPTION:
LIVE OAK CREEK 21.0
END DESCRIPTION:
XS GIS Cut Line= 3
      2745079.85     10055687.28      2744620.54     10055647.59
      2743787.05     10055052.24
#Sta/Elev= 30
  4475.7 1678.21  4487.1 1677.06  4537.3 1675.51  4647.7 1667.45    4687 1663.41
  4707.9 1659.06  4748.1 1652.54  4798.3 1647.78  4908.7 1641.56  4923.6 1639.36
  4935.2 1634.71  4969.3    1632  5040.9  1632.8  5049.5 1634.29  5062.2 1639.01
  5076.5 1642.84  5091.2 1644.07    5106 1643.64  5120.7 1646.56  5141.6 1652.33
  5162.5 1655.37    5192 1657.69  5343.2 1656.35  5485.7 1658.93  5500.5 1660.25
  5515.2 1659.64  5615.2 1662.61    5729 1665.49  5773.3 1665.61    5961 1669.27
#Mann= 4 ,-1 , 0
  4475.7      .1       0  4923.6     .07       0  5076.5      .1       0
  5615.2     .05       0
Bank Sta=4798.3,5120.7
XS Rating Curve= 0 ,0
Exp/Cntr=0.3,0.1

Type RM Length L Ch R = 1 ,11245   ,529,529,529
BEGIN DESCRIPTION:
LIVE OAK CREEK 20.0
END DESCRIPTION:
XS GIS Cut Line= 3
      2745268.51     10055403.75      2744918.47     10055203.73
      2744268.49     10054753.75
#Sta/Elev= 30
    4594 1678.36  4697.7 1674.21  4725.8 1671.67  4778.3 1669.72  4784.8 1666.26
  4806.4 1662.71  4822.2 1658.15  4843.8 1655.45  4893.5 1652.98  4916.5 1645.96
  4930.2  1639.2  4953.6  1635.7  4974.1 1633.71  5016.5 1632.81  5019.2 1632.31
  5022.5 1632.81  5032.1 1633.54  5046.5 1636.38  5070.1 1635.98  5147.8 1640.74
  5198.5  1646.6  5264.1 1653.48  5299.9 1654.48  5622.2 1653.41  5693.8 1658.36
  5729.6 1670.72  5744.5  1675.7  5759.3 1683.24  5769.3 1685.36  5787.7 1690.31
#Mann= 8 ,-1 , 0
    4594     .05       0  4725.8     .16       0  4953.6      .1       0
  5016.5     .07       0  5022.5      .1       0  5032.1     .16       0
  5729.6     .05       0  5769.3      .1       0
Bank Sta=4916.5,5198.5
XS Rating Curve= 0 ,0
Exp/Cntr=0.3,0.1

Type RM Length L Ch R = 1 ,10716   ,692,692,692
BEGIN DESCRIPTION:
LIVE OAK CREEK 19.0
END DESCRIPTION:
XS GIS Cut Line= 3
      2745300.94     10054865.14      2744983.42      10054683.7
      2744263.38     10054712.05
#Sta/Elev= 30
  4564.8 1665.28    4613 1663.38  4809.5 1658.55    4839 1654.99  4860.6 1654.56
  4876.5 1647.73  4882.2 1647.59  4890.1 1643.72  4898.1  1641.2  4903.8 1641.45
  4919.7 1638.08  4925.4 1638.72  4930.5 1634.97  5002.5 1633.36  5005.3 1632.86
  5008.5 1633.36  5059.5  1635.9  5075.6 1639.94  5105.6 1639.42  5175.7 1644.05
  5325.8 1654.28  5385.8 1652.36  5475.9 1652.18  5535.9 1655.92  5545.9 1657.59
  5563.9 1663.83  5568.9 1663.52  5576.3 1667.29    5636 1689.06  5651.1 1690.43
#Mann= 6 ,-1 , 0
  4564.8     .05       0    4613      .1       0  5002.5     .07       0
  5008.5      .1       0  5545.9     .05       0  5576.3      .1       0
Bank Sta=4890.1,5175.7
XS Rating Curve= 0 ,0
Exp/Cntr=0.3,0.1

Type RM Length L Ch R = 1 ,10024   ,642,642,642
BEGIN DESCRIPTION:
LIVE OAK CREEK 18.0
END DESCRIPTION:
XS GIS Cut Line= 3
      2745587.76     10054602.54      2744887.01     10053997.35
      2744063.43     10054211.21
#Sta/Elev= 30
    3791 1664.47  3917.4 1661.49  4136.8 1653.32    4343 1650.74  4406.6 1648.88
  4569.6 1649.14  4662.1 1648.24  4787.7 1649.04  4808.4 1647.81    4829  1648.6
  4843.2 1647.38    4860 1642.69  4878.5 1640.46  4924.3 1636.79  4932.4 1634.25
  4942.7 1633.12  4959.7 1633.26  5040.5 1631.91  5140.6 1640.32  5149.3 1641.12
  5180.3 1646.78  5238.4 1655.43  5243.6 1658.26  5308.7 1662.31  5366.3 1662.15
  5428.3 1667.42  5459.3 1668.42  5510.9 1671.49  5557.7 1676.38  5567.8 1676.48
#Mann= 4 ,-1 , 0
    3791      .1       0  4959.7     .07       0  5149.3      .1       0
  5308.7     .05       0
Bank Sta=4878.5,5140.6
XS Rating Curve= 0 ,0
Exp/Cntr=0.3,0.1

Type RM Length L Ch R = 1 ,9382    ,566,566,566
BEGIN DESCRIPTION:
LIVE OAK CREEK 17.0
END DESCRIPTION:
XS GIS Cut Line= 2
      2745669.65     10054502.42      2744022.98     10052983.11
#Sta/Elev= 30
  3477.8  1663.4    3584 1660.07  3683.2 1653.91  3838.6 1652.76  4001.3 1649.84
    4037 1650.33  4107.4 1648.19  4355.2 1646.83  4411.9 1648.25  4489.5 1646.46
  4730.5 1646.61  4758.4 1645.59    4815 1638.41  4864.9 1632.58  5010.5 1632.46
  5013.3 1631.96  5016.5 1632.46  5140.5 1632.55  5154.7 1634.01  5168.9 1639.53
  5176.3 1642.75  5183.1 1647.47  5211.4 1657.35  5225.6 1659.88  5268.1 1663.85
  5353.2  1663.8  5388.3 1666.33  5459.2 1662.86  5586.8 1661.75  5718.3 1662.34
#Mann= 3 ,-1 , 0
  3477.8     .05       0  5010.5    .033       0  5016.5     .05       0
Bank Sta=4815,5168.9
XS Rating Curve= 0 ,0
Exp/Cntr=0.3,0.1

Type RM Length L Ch R = 1 ,8816    ,835,835,835
BEGIN DESCRIPTION:
LIVE OAK CREEK 16.0
END DESCRIPTION:
XS GIS Cut Line= 4
       2745660.6     10054183.93      2745064.48      10053533.2
      2745078.13     10053251.07      2744734.31     10052947.97
#Sta/Elev= 30
  4024.7  1655.3  4043.6 1654.71  4139.6 1653.86  4182.1 1651.57  4287.7 1649.06
  4309.8 1649.23  4365.9 1646.41  4493.5 1636.29  4613.8 1635.77  4670.5 1633.52
  4705.6 1634.46  4727.2 1633.35  4776.6 1636.41  4840.1 1636.55  4875.8 1632.75
  5003.8 1632.27  5006.5 1631.77  5009.8 1632.27  5097.5 1632.38  5136.9 1637.12
    5167 1644.66  5194.5 1649.09  5208.8 1649.88  5237.2 1647.22    5266 1649.19
  5272.3 1650.36  5392.8 1652.34  5533.7 1657.48  5549.1 1659.07    5648 1660.06
#Mann= 7 ,-1 , 0
  4024.7     .05       0  4043.6      .1       0  4287.7     .05       0
  5003.8    .033       0  5009.8     .05       0    5266      .1       0
  5533.7     .05       0
Bank Sta=4840.1,5136.9
XS Rating Curve= 0 ,0
Exp/Cntr=0.3,0.1
