--- UNT 0085 IN HEWA.prj (project) ---

Proj Title=UNT 0085 IN HEWA Base Level Engineering
Current Plan=p01
Default Exp/Contr=0.3,0.1
English Units
Geom File=g01
Flow File=f01
Plan File=p01
Y Axis Title=Elevation
X Axis Title(PF)=Main Channel Distance
X Axis Title(XS)=Station
BEGIN DESCRIPTION:
UNT 0085 IN HEWA
END DESCRIPTION:
DSS Export Rating Curves= 0
DSS Export Rating Curve Sorted= 0
DSS Export Volume Flow Curves= 0
DXF OffsetX= 0
DXF OffsetY= 0
DXF ScaleX= 1
DXF ScaleY= 10

--- UNT 0085 IN HEWA.p01 (plan) ---

Plan Title=Multiple Run
Short Identifier=Multiple
Geom File=g01
Flow File=f01
Subcritical Flow
K Sum by GR= 0
Std Step Tol= 0.01
Critical Tol= 0.01
Num of Std Step Trials= 20
Max Error Tol= 0.3
Flow Tol Ratio= 0.001
Split Flow NTrial= 30
Split Flow Tol= 0.02
Split Flow Ratio= 0.02
Log Output Level= 0
Friction Slope Method= 1
Unsteady Friction Slope Method= 2
Unsteady Bridges Friction Slope Method= 1
Parabolic Critical Depth
Global Vel Dist=  1 , 1 , 1
Global Log Level= 0
CheckData=True
Encroach Param= -1, 0, 0, 0
BEGIN DESCRIPTION:
Multiple Run
END DESCRIPTION:

--- UNT 0085 IN HEWA.f01 (steady flow) ---

Flow Title=Multiple
Program Version=4.10
Number of Profiles= 7
Profile Names=10-year,25-year,50-year,1pct_min,100-year,1pct_plu,500-year
River Rch & RM=UNT 0085 IN HEWA,Reach-1         ,21960
     970    1399    1765    1624    2196    2970    3399
River Rch & RM=UNT 0085 IN HEWA,Reach-1         ,19838
    1653    2446    3141    2933    3966    5364    6332
River Rch & RM=UNT 0085 IN HEWA,Reach-1         ,13631
    2642    3998    5210    4930    6668    9017   10936
River Rch & RM=UNT 0085 IN HEWA,Reach-1         ,13220
    2642    3998    5210    4930    6668    9017   10936
River Rch & RM=UNT 0085 IN HEWA,Reach-1         ,10045
    3214    4901    6420    6103    8253   11161   13659
River Rch & RM=UNT 0085 IN HEWA,Reach-1         ,6180
    3479    5316    6972    6633    8970   12131   14873
Boundary for River Rch & Prof#=UNT 0085 IN HEWA,Reach-1         , 1
Up Type= 0
Dn Type= 3
Dn Slope=0.002
Boundary for River Rch & Prof#=UNT 0085 IN HEWA,Reach-1         , 2
Up Type= 0
Dn Type= 3
Dn Slope=0.002
Boundary for River Rch & Prof#=UNT 0085 IN HEWA,Reach-1         , 3
Up Type= 0
Dn Type= 3
Dn Slope=0.002
Boundary for River Rch & Prof#=UNT 0085 IN HEWA,Reach-1         , 4
Up Type= 0
Dn Type= 3
Dn Slope=0.002
Boundary for River Rch & Prof#=UNT 0085 IN HEWA,Reach-1         , 5
Up Type= 0
Dn Type= 3
Dn Slope=0.002
Boundary for River Rch & Prof#=UNT 0085 IN HEWA,Reach-1         , 6
Up Type= 0
Dn Type= 3
Dn Slope=0.002
Boundary for River Rch & Prof#=UNT 0085 IN HEWA,Reach-1         , 7
Up Type= 0
Dn Type= 3
Dn Slope=0.002
DSS Import GetInterval= 0
DSS Import GetPeak= 0
DSS Import FillOption= 0

--- UNT 0085 IN HEWA.g01 (geometry) ---

Geom Title=Existing Conditions
Program Version=4.10

River Reach=UNT 0085 IN HEWA,Reach-1
Reach XY= 30
      2631157.12     10087804.19      2631649.67     10087116.64
      2632022.99     10087115.24       2632686.1     10087385.94
      2633316.59     10086588.67      2633239.09     10085668.99
      2633558.88     10084785.17      2633388.15     10084355.81
      2633758.18     10083918.47      2633612.09     10083684.94
      2633765.34     10083507.64      2634137.89     10083511.64
      2634604.76     10083097.91      2634525.82     10082567.28
      2635603.83     10081826.59      2636006.68     10081029.54
      2636569.84     10080756.61       2637200.2     10080700.69
      2637600.01      10080353.4      2638097.88     10077936.29
      2637849.55      10077105.3      2637851.45     10076184.97
       2638009.9     10075877.36      2638762.46     10075881.25
      2639278.47     10075523.73      2639287.59      10075289.1
      2638898.81     10074758.48       2639037.1     10073773.34
      2638920.21     10073339.49      2639936.67     10072658.29

Type RM Length L Ch R = 1 ,21960   ,272,272,272
BEGIN DESCRIPTION:
UNT 0085 IN HEWA 46.0
END DESCRIPTION:
XS GIS Cut Line= 2
      2631551.07      10087830.8      2630895.77     10087237.92
#Sta/Elev= 30
  4745.2 2155.89  4766.1  2154.8  4801.9 2154.13  4822.8 2152.97  4879.6 2151.11
  4886.4 2150.31  4916.5 2148.91  4936.4 2147.79  4964.5 2145.39  4978.3 2141.48
  4989.5 2137.63  4992.2 2137.13  4995.5 2137.63  5006.7 2138.27  5014.1 2139.62
  5056.7  2141.8    5106 2141.46  5212.2 2143.63  5226.3 2144.55  5360.8 2150.28
  5403.4 2152.99  5431.8 2154.08  5452.8 2155.84  5460.2 2155.76  5486.8 2157.06
  5509.5 2158.36    5517 2158.29  5523.7 2158.92  5580.5 2159.72  5628.9 2160.97
#Mann= 5 ,-1 , 0
  4745.2      .1       0  4916.5     .16       0  4989.5     .07       0
  4995.5     .16       0  5486.8      .1       0
Bank Sta=4989.5,4995.5
XS Rating Curve= 0 ,0
Exp/Cntr=0.3,0.1

Type RM Length L Ch R = 1 ,21688   ,564,564,564
BEGIN DESCRIPTION:
UNT 0085 IN HEWA 45.0
END DESCRIPTION:
XS GIS Cut Line= 3
      2631738.72     10087615.89      2631394.96     10087350.26
      2631311.61     10087068.98
#Sta/Elev= 30
  4672.1 2148.55  4681.3 2148.56  4702.1 2147.32  4795.4 2145.24  4847.7 2143.49
    4895 2141.63  4915.8 2139.81  4944.8 2138.38  4988.3 2136.76  4994.6 2137.07
    4998 2135.37  5000.7 2134.87    5004 2135.37  5009.1 2137.31  5044.4 2137.75
  5065.2 2139.17  5079.7 2139.06  5094.2 2139.56  5101.2 2140.17  5143.2 2141.66
  5148.4 2142.37  5163.3 2143.18  5192.7 2144.34  5220.1 2146.29  5248.1 2147.68
  5280.2 2149.86  5291.8  2151.3  5311.5 2152.34  5363.7 2158.77  5399.9 2160.92
#Mann= 6 ,-1 , 0
  4672.1      .1       0  4847.7     .16       0    4998     .07       0
    5004     .16       0  5163.3      .1       0  5192.7     .16       0
Bank Sta=4998,5004
XS Rating Curve= 0 ,0
Exp/Cntr=0.3,0.1

Type RM Length L Ch R = 1 ,21124   ,457,457,457
BEGIN DESCRIPTION:
UNT 0085 IN HEWA 44.0
END DESCRIPTION:
XS GIS Cut Line= 2
       2631819.9     10087485.45      2631793.94     10086820.16
#Sta/Elev= 30
  4616.3 2142.76    4648 2141.46  4658.1 2140.67  4668.1 2139.54  4688.1 2138.22
  4728.1 2137.04  4748.1 2136.04  4800.6  2135.4  4918.2 2134.59  4958.3 2133.39
  4968.3 2132.63  4978.3 2132.37  4995.3 2131.06  4998.1 2130.56  5001.3 2131.06
  5008.3  2131.7  5018.8 2133.37  5028.3 2136.18  5035.6 2139.89  5040.6 2140.27
  5048.3 2142.62  5068.4 2145.34  5078.4 2146.14  5128.4 2151.16  5158.4 2154.85
  5188.5 2157.07  5218.5 2159.79  5228.5 2160.55  5248.5 2161.41  5282.1 2162.05
#Mann= 5 ,-1 , 0
  4616.3      .1       0  4800.6     .16       0  4995.3     .07       0
  5001.3     .16       0  5018.8      .1       0
Bank Sta=4995.3,5001.3
XS Rating Curve= 0 ,0
Exp/Cntr=0.3,0.1

Type RM Length L Ch R = 1 ,20667   ,346,346,346
BEGIN DESCRIPTION:
UNT 0085 IN HEWA 43.0
END DESCRIPTION:
XS GIS Cut Line= 3
      2632218.47     10087553.76      2632218.47     10087253.73
      2632168.46     10087003.71
#Sta/Elev= 30
    4688  2143.4  4690.5  2143.4    4718 2142.18  4739.6 2140.76    4758 2139.48
    4768 2139.25    4778 2138.56    4848 2131.65    4858 2131.06    4878 2130.32
  4938.5 2128.75    4948 2128.26    4965 2126.87  4967.8 2126.37    4971 2126.87
  4998.2 2126.89  5018.6 2127.25    5039 2129.59  5049.2 2130.44  5069.6 2131.57
  5079.8 2132.42  5110.4  2134.6  5130.8 2135.77  5161.4 2138.03  5181.8 2139.83
    5192 2140.58  5202.2 2141.02  5232.8 2141.97  5240.4 2142.38    5243 2142.38
#Mann= 5 ,-1 , 0
    4688      .1       0  4739.6     .16       0  4938.5      .1       0
    4965     .07       0    4971      .1       0
Bank Sta=4965,4971
XS Rating Curve= 0 ,0
Exp/Cntr=0.3,0.1

Type RM Length L Ch R = 1 ,20321   ,483,483,483
BEGIN DESCRIPTION:
UNT 0085 IN HEWA 42.0
END DESCRIPTION:
XS GIS Cut Line= 3
      2632485.24     10087660.68      2632566.37     10087206.33
      2632245.08     10086690.31
#Sta/Elev= 30
    4679 2144.02    4747 2140.71    4808 2138.92    4834 2136.69  4834.3 2136.65
  4879.1  2132.8  4889.2 2131.47  4895.4 2129.67  4909.5 2127.21  4919.7 2126.34
  4980.6 2125.14  4990.8 2123.57    4998 2123.51  5000.7 2123.01    5004 2123.51
  5008.1 2124.19  5013.2 2123.55  5067.1 2127.41  5082.2 2126.66  5120.9 2127.72
  5143.3 2127.12  5190.7  2128.2  5220.9 2129.94  5336.6 2133.56  5388.5 2134.68
  5555.9 2142.68  5567.9 2143.84  5671.8 2147.59  5698.9  2149.8  5748.4 2151.35
#Mann= 5 ,-1 , 0
    4679      .1       0    4834     .16       0  4834.3      .1       0
    4998     .07       0    5004      .1       0
Bank Sta=4998,5004
XS Rating Curve= 0 ,0
Exp/Cntr=0.3,0.1

Type RM Length L Ch R = 1 ,19838   ,416,416,416
BEGIN DESCRIPTION:
UNT 0085 IN HEWA 41.0
END DESCRIPTION:
XS GIS Cut Line= 2
      2633171.52     10087453.69      2632494.47     10086729.76
#Sta/Elev= 30
  4531.7 2149.54  4569.3 2148.39  4604.5 2146.49  4703.7 2143.46  4717.8 2142.83
  4724.7 2141.75    4732 2141.67  4774.5 2138.59  4842.6 2135.78  4887.6 2134.11
    4923 2130.99  4951.3 2126.28  4958.2 2123.95  4972.3 2120.79  4986.5 2119.98
  4997.7 2118.43  5000.4 2117.93  5003.7 2118.43  5014.8 2120.51  5020.3 2120.72
    5029 2121.62  5043.2 2121.89  5128.2 2122.25  5269.8 2126.77  5298.2 2128.72
    5305 2129.65    5326 2130.76  5418.3 2134.17  5516.8  2139.3  5522.9  2139.3
#Mann= 5 ,-1 , 0
  4531.7      .1       0  4842.6     .16       0  4997.7     .07       0
  5003.7     .16       0  5020.3      .1       0
Bank Sta=4997.7,5003.7
XS Rating Curve= 0 ,0
Exp/Cntr=0.3,0.1

Type RM Length L Ch R = 1 ,19422   ,486,486,486
BEGIN DESCRIPTION:
UNT 0085 IN HEWA 40.0
END DESCRIPTION:
XS GIS Cut Line= 3
      2633359.05     10087026.63      2632895.51     10086594.34
      2632614.29     10086479.76
#Sta/Elev= 30
  4626.3 2145.23  4642.7 2145.04  4664.2 2143.97  4671.1 2144.27  4692.6 2141.66
  4706.7 2141.12  4784.4 2135.71  4869.4 2131.02  4876.3 2129.45  4904.6 2119.82
  4911.9 2118.98  4940.3 2119.11  4993.4 2117.54  4996.2 2117.04  4999.4 2117.54
  5032.1 2119.09  5054.6 2119.27  5133.2 2119.77  5260.1 2120.68  5279.5 2121.72
  5289.3 2123.17  5303.5 2124.25  5321.7 2126.46  5327.6 2127.99    5333 2128.72
  5397.3 2131.88  5451.3 2133.22  5494.5 2135.81  5536.2 2137.35  5563.8 2138.96
#Mann= 5 ,-1 , 0
  4626.3      .1       0  4993.4     .07       0  4999.4      .1       0
  5054.6     .16       0  5133.2      .1       0
Bank Sta=4993.4,4999.4
XS Rating Curve= 0 ,0
Exp/Cntr=0.3,0.1

Type RM Length L Ch R = 1 ,18936   ,433,433,433
BEGIN DESCRIPTION:
UNT 0085 IN HEWA 39.0
END DESCRIPTION:
XS GIS Cut Line= 3
      2633629.84     10086427.67      2633166.34     10086396.42
      2632703.16     10086349.58
#Sta/Elev= 30
  4716.8  2138.1  4776.4 2135.35    4824 2133.53  4878.5  2131.3  4898.6 2129.29
  4928.7 2127.55  4952.2 2125.53  4958.7 2125.05  4968.7  2123.2  4978.8 2116.96
  4988.8 2113.01  4993.1 2112.45  4995.8 2111.95  4999.1 2112.45  5028.9 2113.24
  5038.9 2114.46  5084.8 2115.45  5279.7 2117.36  5334.8 2118.35  5361.2 2118.67
  5390.3 2119.82  5420.4 2122.01  5439.3  2124.5  5456.1 2127.52  5480.7 2129.25
  5490.8 2129.25    5556  2131.9  5571.2 2134.15  5581.3 2133.22  5646.9 2135.91
#Mann= 9 ,-1 , 0
  4716.8      .1       0  4776.4     .16       0    4824      .1       0
  4952.2     .16       0  4993.1     .07       0  4999.1     .16       0
  5084.8      .1       0  5334.8     .16       0  5439.3      .1       0
Bank Sta=4993.1,4999.1
XS Rating Curve= 0 ,0
Exp/Cntr=0.3,0.1

Type RM Length L Ch R = 1 ,18503   ,409,409,409
BEGIN DESCRIPTION:
UNT 0085 IN HEWA 38.0
END DESCRIPTION:
XS GIS Cut Line= 3
      2633618.44     10085953.73      2633218.47     10086003.73
      2632968.46     10086003.73
#Sta/Elev= 30
  4619.5 2127.48  4639.6 2126.39  4657.3 2124.76  4662.3 2125.15  4737.9 2115.56
  4742.9 2115.93  4750.5 2115.14  4760.6 2114.59  4777.5 2114.13  4871.4 2112.07
  4911.7 2113.01  4931.9 2112.97    4952    2112  4962.1 2110.59  4972.2 2110.05
  4979.8 2110.05  4999.4    2109  5002.2  2108.5  5005.4    2109  5020.1 2110.77
  5052.6 2112.07  5072.6 2113.95  5102.6  2114.9  5142.6  2115.6  5152.6 2116.14
  5172.6 2117.86  5192.6 2120.59  5222.6 2123.74  5242.6 2125.28  5272.6 2126.97
#Mann= 4 ,-1 , 0
  4619.5     .16       0  4777.5      .1       0  4999.4     .07       0
  5005.4      .1       0
Bank Sta=4999.4,5005.4
XS Rating Curve= 0 ,0
Exp/Cntr=0.3,0.1

Type RM Length L Ch R = 1 ,18094   ,419,419,419
BEGIN DESCRIPTION:
UNT 0085 IN HEWA 37.0
END DESCRIPTION:
XS GIS Cut Line= 3
      2633668.49     10085703.74      2633268.47     10085603.73
      2633018.46     10085653.73
#Sta/Elev= 30
    4591 2125.17  4601.3 2124.65    4622 2122.59  4650.3 2120.43  4663.2 2119.76
  4683.8 2116.27  4691.5 2113.42  4704.4 2112.11    4756 2110.79  4811.1  2110.6
  4879.6 2110.44  4944.1  2109.4  4972.4 2107.33  4980.1 2105.48  4985.3 2105.16
    4990  2104.1  4992.8  2103.6    4996  2104.1  5000.8 2104.99  5013.5 2105.32
  5033.9 2107.17  5044.1 2110.87  5054.3  2112.4  5084.9 2113.29  5115.5 2113.63
  5146.1 2114.69  5176.7 2117.02  5190.1  2118.8  5248.1 2121.78  5258.3  2122.6
#Mann= 5 ,-1 , 0
    4591     .16       0  4811.1      .1       0    4990     .07       0
    4996      .1       0  5190.1      .1       0
Bank Sta=4990,4996
XS Rating Curve= 0 ,0
Exp/Cntr=0.3,0.1

Type RM Length L Ch R = 1 ,17675   ,481,481,481
BEGIN DESCRIPTION:
UNT 0085 IN HEWA 36.0
END DESCRIPTION:
XS GIS Cut Line= 3
       2633668.5     10085303.74      2633368.47     10085203.73
      2632968.44     10085253.74
#Sta/Elev= 30
  4701.6 2119.68  4723.7  2119.2  4743.8 2118.71  4754.3 2117.91  4832.5 2114.51
  4870.3 2112.63  4880.8 2111.02  4901.9  2106.3  4912.5 2105.39  4975.7 2106.08
  4986.2 2104.36  4993.8 2102.41  4996.5 2101.91  4999.8 2102.41  5015.2 2104.33
  5027.9 2104.55  5048.1 2105.77  5078.3 2106.13  5118.6 2105.65    5169 2106.77
  5216.9 2107.13    5244    2108    5290 2111.81  5297.5 2112.97  5302.6 2113.09
  5310.1 2114.11  5333.4    2116  5360.5 2117.87  5383.2 2118.72    5421 2121.57
#Mann= 7 ,-1 , 0
  4701.6      .1       0  4723.7     .16       0  4832.5      .1       0
  4993.8     .07       0  4999.8      .1       0    5244     .16       0
  5333.4      .1       0
Bank Sta=4993.8,4999.8
XS Rating Curve= 0 ,0
Exp/Cntr=0.3,0.1

Type RM Length L Ch R = 1 ,17194   ,473,473,473
BEGIN DESCRIPTION:
UNT 0085 IN HEWA 35.0
END DESCRIPTION:
XS GIS Cut Line= 3
      2633993.93     10085079.43      2633624.12     10084756.51
      2632863.73     10085032.54
#Sta/Elev= 30
  4439.6 2127.13    4518 2125.34  4546.8 2124.94  4659.7 2116.55  4730.9 2113.16
  4773.6 2109.11  4919.2 2105.29  4934.2 2104.76  4947.2 2102.31  4957.9 2101.42
  4979.1 2101.28  4997.7 2099.77  5000.5 2099.27  5003.7 2099.77    5011 2101.12
  5044.1 2102.22  5064.2 2102.09  5074.9 2101.08  5117.8 2103.08    5160 2101.93
    5235  2103.2  5308.9 2102.91    5394 2103.81  5438.6 2104.98  5500.4 2109.04
  5525.1 2109.83  5611.6 2116.49  5636.9 2119.68  5698.1 2123.83  5739.5 2124.16
#Mann= 6 ,-1 , 0
  4439.6     .16       0    4518      .1       0  4919.2     .16       0
  4997.7     .07       0  5003.7     .16       0  5044.1      .1       0
Bank Sta=4997.7,5003.7
XS Rating Curve= 0 ,0
Exp/Cntr=0.3,0.1

Type RM Length L Ch R = 1 ,16721   ,80,80,80
BEGIN DESCRIPTION:
UNT 0085 IN HEWA 34.0
END DESCRIPTION:
XS GIS Cut Line= 3
      2633886.15     10084891.58      2633375.71     10084388.09
      2632663.88     10083829.04
#Sta/Elev= 30
  4296.9 2118.61  4392.7    2112  4456.4 2108.98  4682.7 2103.05  4802.8 2100.73
  4845.3 2101.11  4873.6 2099.92  4887.7 2099.96    4916 2103.49  4930.1 2102.14
  4951.4 2096.35  4983.7 2094.25  4986.5 2093.75  4989.7 2094.25  5099.8 2096.47
  5122.3 2097.88  5143.1 2101.31  5157.6 2100.29  5192.8 2102.62  5370.9 2102.79
  5484.8 2105.28  5492.9 2106.55  5534.5 2105.74  5691.7 2107.81  5791.2 2116.68
  5805.6  2116.5    5812 2118.31  5820.1 2118.54  5840.9 2121.79    5919 2124.29
#Mann= 3 ,-1 , 0
  4296.9      .1       0  4983.7     .07       0  4989.7      .1       0
Bank Sta=4983.7,4989.7
XS Rating Curve= 0 ,0
Exp/Cntr=0.3,0.1

Type RM Length L Ch R = 1 ,16641   ,61,61,61
BEGIN DESCRIPTION:
Mapping XS 1aa1fac5
END DESCRIPTION:
XS GIS Cut Line= 3
      2633896.53      10084797.8      2633424.32       10084336.
      2632809.76     10083853.38
#Sta/Elev= 30
  4328.1  2114.8  4478.2 2107.92  4584.2  2104.8  4913.5 2098.95  4916.3 2098.45
  4919.5 2098.95  4923.7    2101  4930.7 2100.61  4937.8 2102.82  5001.4 2105.06
  5015.8 2102.24  5022.2 2104.48  5030.3 2102.49  5036.6 2104.78  5044.7 2103.12
  5051.1 2105.05  5059.2 2104.05  5065.5 2105.22  5094.4 2105.36  5100.8 2103.55
  5108.9 2103.78  5115.3 2101.74  5129.7 2102.18  5136.1  2100.8  5158.6 2102.53
  5378.3 2102.46  5442.5 2105.26  5521.1 2104.88  5643.1 2109.89    5770 2121.24
#Mann= 3 ,-1 , 0
  4328.1      .1       0  4913.5     .07       0  4919.5      .1       0
Bank Sta=4913.5,4919.5
XS Rating Curve= 0 ,0
Exp/Cntr=0.3,0.1

Type RM Length L Ch R = 1 ,16580   ,305,305,305
BEGIN DESCRIPTION:
Mapping XS 40041dd1
END DESCRIPTION:
XS GIS Cut Line= 2
      2634031.95     10084780.44      2632886.14     10083794.35
#Sta/Elev= 30
    4243 2122.25  4313.6 2116.56  4413.4  2111.6  4448.5 2108.94  4491.3 2107.41
  4675.6 2102.68  4867.6 2099.93  4909.3 2098.06  4952.1 2097.91  4963.4 2096.78
  4966.1 2096.28  4969.4 2096.78  5023.4 2097.56  5058.6 2096.85  5087.1 2098.78
  5150.7 2099.35    5222 2101.77  5320.8 2101.55    5470 2103.44  5512.8 2105.64
  5533.7 2108.02  5547.9 2108.22  5554.5 2109.67    5583 2111.78  5625.8 2113.99
  5654.3 2114.02  5675.2 2117.17  5682.9 2116.66  5703.7  2119.1  5754.7 2121.74
#Mann= 3 ,-1 , 0
    4243      .1       0  4963.4     .07       0  4969.4      .1       0
Bank Sta=4963.4,4969.4
XS Rating Curve= 0 ,0
Exp/Cntr=0.3,0.1

Type RM Length L Ch R = 1 ,16275   ,714,714,714
BEGIN DESCRIPTION:
UNT 0085 IN HEWA 33.0
END DESCRIPTION:
XS GIS Cut Line= 2
      2634170.82     10084599.86      2633182.35     10083552.43
#Sta/Elev= 30
  4262.9 2119.64  4311.5 2117.32    4375 2112.72  4452.7 2109.01  4502.5 2107.74
  4580.1 2103.16  4778.4 2098.82  4813.6  2098.9  4926.9  2096.6    4962 2097.11
  4983.5 2095.78  4994.7 2093.48  4997.4 2092.98  5000.7 2093.48  5011.8 2094.76
  5117.8 2095.34  5167.2 2097.15  5287.7 2096.46    5344 2097.11  5351.2 2095.78
  5379.6 2097.16    5422 2097.62  5464.5 2099.78  5492.8 2102.52    5528 2109.39
  5542.2 2110.71    5613 2114.72  5676.5 2120.89  5690.7 2121.71  5703.1 2121.31
#Mann= 3 ,-1 , 0
  4262.9      .1       0  4994.7     .07       0  5000.7      .1       0
Bank Sta=4994.7,5000.7
XS Rating Curve= 0 ,0
Exp/Cntr=0.3,0.1

Type RM Length L Ch R = 1 ,15561   ,307,307,307
BEGIN DESCRIPTION:
UNT 0085 IN HEWA 32.0
END DESCRIPTION:
XS GIS Cut Line= 3
      2634197.02     10084381.47      2633707.46     10083391.92
      2633275.21     10083277.35
#Sta/Elev= 30
  4025.3 2110.62  4089.7 2107.97  4156.7 2106.44  4232.7  2101.7  4283.2 2100.02
  4491.4  2095.3  4664.5 2093.04  4770.3 2093.73  4888.8 2091.61  4926.5 2091.68
  4948.8 2090.58  4978.6 2090.96    4998 2089.33  5000.8 2088.83    5004 2089.33
  5015.7 2092.18    5029 2093.73  5068.3 2094.48    5211 2100.79  5231.7 2103.18
  5252.4 2104.65  5263.4 2106.84  5298.4 2108.82  5304.2 2109.71  5355.9 2111.63
  5438.6 2116.52  5454.1 2116.02  5469.7 2118.34  5500.7 2120.72  5576.5 2124.29
#Mann= 3 ,-1 , 0
  4025.3      .1       0    4998     .07       0    5004      .1       0
Bank Sta=4998,5004
XS Rating Curve= 0 ,0
Exp/Cntr=0.3,0.1

Type RM Length L Ch R = 1 ,15254   ,623,623,623
BEGIN DESCRIPTION:
UNT 0085 IN HEWA 31.0
END DESCRIPTION:
XS GIS Cut Line= 3
      2634306.42     10084313.81      2634019.96      10083376.3
      2633296.01     10083001.31
#Sta/Elev= 30
  4173.5 2109.25    4214 2107.73  4299.1 2106.31  4388.4 2100.62  4508.2  2099.2
  4797.7 2090.83  4835.7 2090.56  4947.4 2091.94  4972.1 2090.51  4989.2 2086.48
  4996.6 2085.99  4999.4 2085.49  5002.6 2085.99  5004.9 2087.88  5037.7 2089.79
  5103.3 2089.03  5335.7 2093.91  5431.3  2096.7  5475.5 2099.08  5504.6 2101.69
  5564.1 2103.67  5580.6 2105.59  5602.7  2105.2  5630.5  2109.6    5647 2110.79
  5757.6 2115.43    5824  2119.2  5898.8 2124.89  5906.9 2126.22  5969.1  2128.3
#Mann= 3 ,-1 , 0
  4173.5      .1       0  4996.6     .07       0  5002.6      .1       0
Bank Sta=4996.6,5002.6
XS Rating Curve= 0 ,0
Exp/Cntr=0.3,0.1

Type RM Length L Ch R = 1 ,14631   ,414,414,414
BEGIN DESCRIPTION:
UNT 0085 IN HEWA 30.0
END DESCRIPTION:
XS GIS Cut Line= 3
      2634439.67     10084120.09      2634674.05      10083291.1
      2633793.21     10082744.37
#Sta/Elev= 30
    3933  2100.7  4074.7 2098.57  4116.3 2099.17  4137.1 2098.03    4189 2097.06
  4563.1  2092.2    4604 2090.22  4609.2 2090.45  4615.1 2089.51  4643.2 2088.02
  4677.2 2087.21  4793.4 2086.81  4870.3 2085.81  4897.4  2084.8  4964.8 2085.57
  4998.1 2084.61  5000.9 2084.11  5004.1 2084.61  5043.9 2086.27  5159.6 2086.49
  5290.7 2088.36    5364 2088.63  5558.8 2093.37  5637.9 2096.46  5674.6 2098.72
  5726.5 2100.25  5777.9 2103.13  5784.4 2104.61    5821 2105.55  5831.2 2107.87
#Mann= 3 ,-1 , 0
    3933      .1       0  4998.1     .07       0  5004.1      .1       0
Bank Sta=4998.1,5004.1
XS Rating Curve= 0 ,0
Exp/Cntr=0.3,0.1

Type RM Length L Ch R = 1 ,14217   ,586,586,586
BEGIN DESCRIPTION:
UNT 0085 IN HEWA 29.0
END DESCRIPTION:
XS GIS Cut Line= 3
       2634808.6      10083790.2      2634799.92      10082956.9
      2633753.89     10082653.07
#Sta/Elev= 30
  3886.5 2092.23    4003 2092.17    4233 2090.11    4693 2084.42  4753.5 2084.11
  4835.9 2085.44  4854.1  2084.5  4859.3    2085  4887.6 2082.94  4959.9 2082.68
  5000.9  2080.6  5003.7  2080.1  5006.9  2080.6  5023.3 2082.67  5032.2 2082.43
  5037.4 2083.69    5065 2082.97  5104.5 2084.51  5210.4    2087  5314.9 2088.76
  5523.2 2096.04  5554.4 2098.25  5564.8 2098.53  5577.1 2097.77  5616.9 2101.34
  5637.7 2102.21  5649.4 2103.86  5682.9 2106.75  5741.9 2108.66  5809.1 2112.32
#Mann= 3 ,-1 , 0
  3886.5      .1       0  5000.9     .07       0  5006.9      .1       0
Bank Sta=5000.9,5006.9
XS Rating Curve= 0 ,0
Exp/Cntr=0.3,0.1

Type RM Length L Ch R = 1 ,13631   ,411,411,411
BEGIN DESCRIPTION:
UNT 0085 IN HEWA 28.0
END DESCRIPTION:
XS GIS Cut Line= 3
      2635736.03     10083217.06      2634584.96     10082295.17
      2633632.66     10082456.48
#Sta/Elev= 30
  3721.8 2123.67  3744.3 2123.79  3829.3 2118.48  3885.4 2110.17    3943 2104.74
  4021.4    2091    4071 2086.37  4277.5 2082.46  4298.3 2080.78  4391.1 2081.32
  4405.6 2083.41  4490.4 2081.55  4661.6 2081.98  4711.3 2078.21  4725.7 2080.13
  4882.5 2080.23  4946.5 2077.43  4981.8 2078.09  4999.6 2074.36  5002.3 2073.86
  5005.6 2074.36  5031.4 2082.49    5089 2085.79  5314.7 2088.01    5548 2094.08
  5568.3 2093.51  5720.4 2098.99  5781.2  2102.6  5992.7 2107.05  6162.4 2113.91
#Mann= 3 ,-1 , 0
  3721.8      .1       0  4999.6     .07       0  5005.6      .1       0
#XS Ineff= 2 , 0
         4402.61 2083.24
Permanent Ineff=
       F       F
Bank Sta=4999.6,5005.6
XS Rating Curve= 0 ,0
Exp/Cntr=0.3,0.1

Type RM Length L Ch R = 1 ,13220   ,401,401,401
BEGIN DESCRIPTION:
UNT 0085 IN HEWA 27.0
END DESCRIPTION:
XS GIS Cut Line= 3
      2635724.35     10082991.28      2634979.59     10082111.11
      2634636.55      10081487.4
#Sta/Elev= 30
  3953.2 2108.94  3976.4 2106.11  3984.1  2103.7  3990.7 2102.89  3998.4 2100.03
    4027 2094.67  4062.1  2090.3  4097.3 2088.44  4281.9 2085.82  4423.6 2087.02
  4501.6 2085.99  4615.9  2082.2  4665.3    2079  4842.2 2077.47  4906.3 2075.49
  4956.5 2076.67  4970.8 2074.98  4995.2 2070.64  4997.9 2070.14  5001.2 2070.64
  5005.9 2070.79  5026.7 2076.52  5244.6 2078.85    5320 2078.87  5377.1 2081.77
  5472.9 2084.77  5510.7 2086.67  5673.6 2090.73  5685.2 2091.69    5818 2096.35
#Mann= 3 ,-1 , 0
  3953.2      .1       0  4995.2     .07       0  5001.2      .1       0
Bank Sta=4995.2,5001.2
XS Rating Curve= 0 ,0
Exp/Cntr=0.3,0.1

Type RM Length L Ch R = 1 ,12819   ,458,458,458
BEGIN DESCRIPTION:
UNT 0085 IN HEWA 26.0
END DESCRIPTION:
XS GIS Cut Line= 3
      2635718.48     10082303.74      2635318.47     10081903.73
      2634852.12     10081431.07
#Sta/Elev= 30
  4444.2 2086.74  4659.4 2079.22  4669.1 2078.76  4712.9  2075.2  4797.8 2074.41
  4868.5 2073.01    4925 2073.89  4967.5 2073.21  4981.6 2072.61  4992.8 2070.64
  4995.5 2070.14  4998.8 2070.64  5006.4 2071.67  5013.4 2071.67  5031.1 2073.88
  5038.1 2074.08  5200.8  2077.1    5222 2077.02  5271.5 2078.34  5285.7 2078.93
  5306.9 2081.09  5328.1 2082.34  5335.1 2083.31  5391.7 2086.67  5427.1 2087.43
  5504.9 2090.07  5547.3 2092.43  5589.7 2093.59  5639.3 2096.07  5673.9  2097.2
#Mann= 5 ,-1 , 0
  4444.2      .1       0  4659.4     .16       0  4669.1      .1       0
  4992.8     .07       0  4998.8      .1       0
Bank Sta=4992.8,4998.8
XS Rating Curve= 0 ,0
Exp/Cntr=0.3,0.1

Type RM Length L Ch R = 1 ,12361   ,371,371,371
BEGIN DESCRIPTION:
UNT 0085 IN HEWA 25.0
END DESCRIPTION:
XS GIS Cut Line= 3
      2635868.47     10082153.74      2635668.47     10081703.73
      2635268.49     10081303.76
#Sta/Elev= 30
  4474.2 2085.78  4558.3 2083.27  4594.6  2081.1  4627.4 2079.87  4649.3 2078.36
  4693.1 2073.61  4708.8 2072.65  4747.8 2071.99    4784 2072.39  4809.9 2072.15
  4859.3 2072.27  4868.2  2071.8  4877.1 2070.69  4882.5 2069.43  4890.1  2068.6
  4900.3  2068.9  4911.9 2070.13  4934.5 2070.86  4970.2 2070.44  4991.9 2065.31
  4994.7 2064.81  4997.9 2065.31  5027.2 2067.85  5051.5 2071.18  5122.2 2071.95
  5263.6 2074.46  5334.3 2076.49  5390.9 2078.52  5433.3 2081.65  5532.3 2085.77
#Mann= 5 ,-1 , 0
  4474.2      .1       0  4809.9     .16       0  4991.9     .07       0
  4997.9     .16       0  5027.2      .1       0
Bank Sta=4991.9,4997.9
XS Rating Curve= 0 ,0
Exp/Cntr=0.3,0.1

Type RM Length L Ch R = 1 ,11990   ,421,421,421
BEGIN DESCRIPTION:
UNT 0085 IN HEWA 24.0
END DESCRIPTION:
XS GIS Cut Line= 2
       2636353.9     10081815.65      2635458.05     10081018.75
#Sta/Elev= 30
  4383.1 2081.42    4417  2080.7  4523.2 2076.74  4544.1    2075  4558.3 2074.69
  4593.5 2072.41  4671.4 2070.72  4728.1 2068.69  4784.9 2067.47  4799.2 2067.83
  4805.9 2068.76  4891.1 2067.52  4933.8  2068.3  4968.9 2067.52  4976.4 2067.02
  4994.3 2061.18  4997.1 2060.68  5000.3 2061.18  5011.6  2062.9  5019.1 2065.57
  5032.8 2066.64  5082.6 2066.25  5111.1 2067.79  5223.9 2070.93  5245.7 2072.92
  5287.5 2079.39  5351.9 2084.63  5521.6 2088.62  5556.7  2090.2  5582.1  2090.4
#Mann= 3 ,-1 , 0
  4383.1      .1       0  4994.3     .07       0  5000.3      .1       0
Bank Sta=4994.3,5000.3
XS Rating Curve= 0 ,0
Exp/Cntr=0.3,0.1

Type RM Length L Ch R = 1 ,11569   ,501,501,501
BEGIN DESCRIPTION:
UNT 0085 IN HEWA 23.0
END DESCRIPTION:
XS GIS Cut Line= 2
      2636428.62     10081800.42      2635780.94     10080560.38
#Sta/Elev= 30
  4123.2 2081.99  4277.4 2077.01  4344.9 2073.26  4378.9 2070.28  4411.1  2069.2
  4469.2 2068.69  4549.3 2066.77    4654 2065.67  4852.8 2064.25  4891.3 2064.88
  4920.5 2064.61  4957.5 2063.51    4974 2062.48  4979.6 2061.28  4988.2  2060.5
  4998.7 2056.19  5001.5 2055.69  5004.7 2056.19  5010.7 2060.28  5018.2  2067.7
  5033.3 2073.97  5045.9 2076.24    5068 2078.09  5106.5 2079.74  5255.4 2083.29
  5261.1 2083.94  5305.2 2085.43  5349.4 2086.23  5426.4 2086.53  5522.2 2088.39
#Mann= 3 ,-1 , 0
  4123.2      .1       0  4998.7     .07       0  5004.7      .1       0
Bank Sta=4998.7,5004.7
XS Rating Curve= 0 ,0
Exp/Cntr=0.3,0.1

Type RM Length L Ch R = 1 ,11068   ,463,463,463
BEGIN DESCRIPTION:
UNT 0085 IN HEWA 22.0
END DESCRIPTION:
XS GIS Cut Line= 3
      2636868.45     10081603.69      2636468.47     10080803.73
      2636268.45     10080653.72
#Sta/Elev= 30
  4103.6 2080.19  4162.3 2077.56  4201.4 2074.99    4207    2075  4251.7 2072.11
  4268.5 2070.12  4290.8 2068.52  4313.2 2067.79  4318.8 2068.03  4357.9 2066.61
  4581.5 2062.92  4849.8 2061.63  4872.2 2060.71  4930.9 2061.03  4967.2  2059.9
    4984 2057.89  4992.2 2057.32  4994.9 2056.82  4998.2 2057.32  5019.9 2058.17
  5026.1  2059.9  5034.4 2061.24  5040.7 2063.92  5055.3 2066.65  5061.5 2067.16
  5134.4 2070.65  5211.5 2073.11  5234.4 2074.36  5244.9 2075.99    5248 2075.99
#Mann= 3 ,-1 , 0
  4103.6      .1       0  4992.2     .07       0  4998.2      .1       0
Bank Sta=4992.2,4998.2
XS Rating Curve= 0 ,0
Exp/Cntr=0.3,0.1

Type RM Length L Ch R = 1 ,10605   ,560,560,560
BEGIN DESCRIPTION:
UNT 0085 IN HEWA 21.0
END DESCRIPTION:
XS GIS Cut Line= 3
      2637016.05     10081605.92      2636901.47     10080652.77
      2636323.43     10080329.91
#Sta/Elev= 30
  4150.6 2081.62  4213.2 2079.59  4257.3 2076.93  4354.2 2068.54  4384.5 2067.27
    4465 2065.42  4837.6 2059.34  4948.5  2059.2  4968.6 2057.22  4988.8 2056.44
  4995.9 2054.17  4998.6 2053.67  5001.9 2054.17    5007 2056.41    5019  2058.6
  5029.1 2058.63  5039.1 2056.24  5079.4 2057.87  5114.8 2058.21  5135.3 2059.37
  5319.2 2062.18  5367.7 2063.92    5422  2065.1  5540.4 2070.21    5618 2073.85
  5676.8 2075.43  5692.8 2077.09  5714.5 2075.81    5744 2077.85  5772.7 2078.82
#Mann= 5 ,-1 , 0
  4150.6      .1       0  4995.9     .07       0  5001.9      .1       0
  5367.7     .05       0  5540.4      .1       0
Bank Sta=4995.9,5001.9
XS Rating Curve= 0 ,0
Exp/Cntr=0.3,0.1

Type RM Length L Ch R = 1 ,10045   ,322,322,322
BEGIN DESCRIPTION:
UNT 0085 IN HEWA 20.0
END DESCRIPTION:
XS GIS Cut Line= 3
      2637984.76     10080715.26      2637495.22     10080579.86
      2636073.39     10079939.25
#Sta/Elev= 30
  4401.7 2079.05  4546.8 2068.99  4577.8    2068  4709.1 2060.14  4836.5 2058.31
  4909.6 2057.76  4940.6 2055.19  4986.9 2053.53  5056.3 2054.67  5084.9 2050.58
    5105 2049.48  5107.8 2048.98    5111 2049.48  5131.2  2050.5  5169.3  2057.2
  5177.5 2057.81  5191.2 2056.68  5246.1 2056.66  5304.1  2058.2  5333.8 2060.16
  5350.4 2059.44  5517.9 2063.27  5765.7 2067.14  5886.9  2070.3  6036.7 2076.31
  6046.7 2077.74  6068.7 2076.28  6090.6 2078.04  6250.5 2084.28  6469.1 2090.87
#Mann= 5 ,-1 , 0
  4401.7      .1       0  4546.8     .05       0  4836.5      .1       0
    5105     .07       0    5111      .1       0
Bank Sta=5105,5111
XS Rating Curve= 0 ,0
Exp/Cntr=0.3,0.1

Type RM Length L Ch R = 1 ,9723    ,483,483,483
BEGIN DESCRIPTION:
UNT 0085 IN HEWA 19.0
END DESCRIPTION:
XS GIS Cut Line= 3
      2638018.46     10080353.73      2637618.47     10080303.73
      2636418.48     10079903.74
#Sta/Elev= 30
  4586.7 2081.85  4616.9 2078.83  4687.5 2069.01  4748.6 2062.52  4785.7 2059.48
  4828.6 2056.85  4969.7    2053  5000.3 2050.41    5032 2051.89  5074.1  2052.7
  5115.6 2050.45  5123.8 2050.37  5126.6 2049.87  5129.8 2050.37    5169 2052.19
  5190.1 2052.26  5221.7 2054.73  5253.3 2054.51  5318.7 2055.52  5389.3  2056.6
  5537.9 2059.86    5559 2061.17  5590.6  2060.7    5812 2064.49  5980.7 2068.69
  6012.3 2069.59  6043.9 2071.12    6065 2072.85  6075.5 2072.72  6254.7 2080.73
#Mann= 7 ,-1 , 0
  4586.7      .1       0  4748.6     .05       0  5115.6      .1       0
  5123.8    .035       0  5129.8      .1       0  5318.7     .05       0
  5389.3      .1       0
Bank Sta=5123.8,5129.8
XS Rating Curve= 0 ,0
Exp/Cntr=0.3,0.1

Type RM Length L Ch R = 1 ,9240    ,457,457,457
BEGIN DESCRIPTION:
UNT 0085 IN HEWA 18.0
END DESCRIPTION:
XS GIS Cut Line= 3
      2638042.08     10080022.56      2637682.72     10079829.86
      2636594.17     10079746.52
#Sta/Elev= 30
  4640.5 2072.36  4649.4 2072.21  4665.7 2069.64  4687.6 2068.08  4775.3 2066.64
  4848.8 2061.58  4857.4 2059.33    4863    2059  4879.3 2054.74  4894.2 2052.92
  4906.9 2051.81    4967  2049.8  4993.4 2045.11  4996.1 2044.61  4999.4 2045.11
  5027.1  2047.6  5072.6 2049.86  5132.8  2050.3  5206.1    2052  5314.9 2053.45
  5604.1 2057.06  5754.6 2060.88  5774.6 2062.69  5794.7 2061.58  5849.4 2062.92
  5980.1 2066.94  6095.6    2072  6105.6 2073.01  6110.8 2075.24    6140 2074.25
#Mann= 5 ,-1 , 0
  4640.5      .1       0  4993.4     .07       0  4999.4      .1       0
  5206.1     .05       0  5314.9      .1       0
Bank Sta=4993.4,4999.4
XS Rating Curve= 0 ,0
Exp/Cntr=0.3,0.1

Type RM Length L Ch R = 1 ,8783    ,424,424,424
BEGIN DESCRIPTION:
UNT 0085 IN HEWA 17.0
END DESCRIPTION:
XS GIS Cut Line= 3
      2638118.48     10079453.73      2637768.47     10079403.73
      2636568.49     10079503.73
#Sta/Elev= 30
  4667.9 2065.88  4728.5 2064.16  4799.2 2060.37  4890.1 2049.53  4960.9 2046.24
  4991.2 2042.51  4998.3 2042.44    5001 2041.94  5004.3 2042.44  5018.9 2044.61
  5051.6 2046.33  5084.2  2046.4  5131.8 2045.08  5151.9 2047.63  5204.6  2048.4
  5272.3  2051.3  5402.8 2052.06  5573.4 2054.92  5844.3 2061.85  5864.4 2063.83
  5884.4 2062.38  5894.5 2062.61    6035 2067.52  6042.5 2068.42  6065.1 2068.55
  6085.1 2065.61  6105.2 2065.11  6125.3 2070.98  6135.3 2071.94  6225.6 2075.87
#Mann= 3 ,-1 , 0
  4667.9      .1       0  4998.3     .07       0  5004.3      .1       0
Bank Sta=4998.3,5004.3
XS Rating Curve= 0 ,0
Exp/Cntr=0.3,0.1

Type RM Length L Ch R = 1 ,8359    ,438,438,438
BEGIN DESCRIPTION:
UNT 0085 IN HEWA 16.0
END DESCRIPTION:
XS GIS Cut Line= 3
      2638168.46     10079203.73      2637918.47     10079003.73
      2636718.47     10078803.73
#Sta/Elev= 30
  4679.9 2063.53  4736.7 2059.81  4815.2 2051.86  4850.4 2050.33  4879.2 2047.91
  4928.8 2045.41  4943.2 2043.85  4993.8 2041.28  4996.6 2040.78  4999.8 2041.28
  5040.6 2044.47  5060.9 2045.11  5088.8 2044.63  5131.8 2042.41  5154.7 2042.13
  5162.3 2042.55  5182.5 2046.73  5192.7  2048.2  5202.8  2048.5  5276.3 2048.43
  5567.8 2051.64  5608.3 2053.23  5762.9 2056.47  5851.6 2059.98  6006.2 2063.64
    6024 2064.28  6044.3  2066.3    6062 2064.18  6094.9 2066.58  6216.6 2070.43
#Mann= 3 ,-1 , 0
  4679.9      .1       0  4993.8     .07       0  4999.8      .1       0
Bank Sta=4993.8,4999.8
XS Rating Curve= 0 ,0
Exp/Cntr=0.3,0.1

Type RM Length L Ch R = 1 ,7921    ,244,244,244
BEGIN DESCRIPTION:
UNT 0085 IN HEWA 15.0
END DESCRIPTION:
XS GIS Cut Line= 3
      2638417.06     10078829.84      2638068.13     10078585.06
      2636683.05      10078538.2
#Sta/Elev= 30
  4494.2 2063.27  4524.1 2062.23  4583.6 2060.18  4629.1 2057.94  4669.9 2055.82
  4712.4 2052.03  4848.6 2048.67  4922.8 2045.11  4997.1 2038.69  4999.9 2038.19
  5003.1 2038.69  5030.2 2042.17  5040.2 2042.59  5070.2 2042.99  5140.2 2040.58
  5190.2 2041.42  5220.3 2044.54  5240.3 2044.14  5290.3 2044.76  5350.3  2044.7
  5470.4 2046.48  5600.5 2050.86  5760.6 2057.25  5940.7 2062.98  6040.7 2064.31
  6120.8 2067.03  6150.8 2067.16  6180.8 2068.53  6250.9 2070.07  6306.3 2072.05
#Mann= 5 ,-1 , 0
  4494.2      .1       0  4524.1     .16       0  4629.1      .1       0
  4997.1     .07       0  5003.1      .1       0
Bank Sta=4997.1,5003.1
XS Rating Curve= 0 ,0
Exp/Cntr=0.3,0.1

Type RM Length L Ch R = 1 ,7677    ,602,602,602
BEGIN DESCRIPTION:
UNT 0085 IN HEWA 14.0
END DESCRIPTION:
XS GIS Cut Line= 2
      2638635.11     10078408.71      2637176.75     10078252.46
#Sta/Elev= 30
  4364.5 2056.01  4391.3 2056.64    4512 2055.39  4542.2 2054.72  4602.5 2051.53
  4632.7 2050.43  4845.5 2046.86  4921.6 2043.78  4984.7 2039.07  5001.8 2038.89
  5004.5 2038.39  5007.8 2038.89  5014.8 2039.17  5020.6  2040.2  5055.1 2040.85
  5125.5 2039.73  5135.5 2040.12  5175.8 2039.62  5195.9 2042.57  5239.1 2042.66
  5307.3 2043.02  5336.7 2042.46    5404  2043.5  5447.3 2043.94  5542.9 2047.76
    5568 2048.98  5583.8 2050.46  5673.5 2053.83  5688.7 2053.95  5831.2 2058.57
#Mann= 9 ,-1 , 0
  4364.5      .1       0  4845.5     .16       0  4921.6      .1       0
  5001.8     .07       0  5007.8      .1       0  5239.1     .05       0
    5404      .1       0  5542.9     .05       0  5673.5      .1       0
Bank Sta=5001.8,5007.8
XS Rating Curve= 0 ,0
Exp/Cntr=0.3,0.1

Type RM Length L Ch R = 1 ,7075    ,363,363,363
BEGIN DESCRIPTION:
UNT 0085 IN HEWA 13.0
END DESCRIPTION:
XS GIS Cut Line= 3
       2638668.5     10077803.73      2638068.47     10077753.73
      2637068.51     10078153.72
#Sta/Elev= 30
  4363.7 2057.49  4405.3 2056.38  4489.2 2053.35  4564.4 2051.09  4684.8 2045.18
  4865.5 2041.11  4903.1 2038.96  4980.6 2036.73  4995.1 2034.41  4997.9 2033.91
  5001.1 2034.41  5057.1 2037.15  5064.1 2037.01  5082.9 2038.37  5142.2 2039.52
  5254.1 2039.23  5333.3 2039.57  5387.2 2041.47    5406 2042.74  5411.4 2042.43
  5435.7  2044.1  5465.3 2044.63  5489.5 2046.32  5645.4 2049.78  5704.9 2052.84
    5763 2053.62  5967.5 2058.05  5974.2 2058.73  6021.3 2059.49  6042.8 2060.48
#Mann= 9 ,-1 , 0
  4363.7      .1       0  4405.3     .16       0  4489.2      .1       0
  4995.1     .07       0  5001.1      .1       0  5057.1     .05       0
  5254.1      .1       0  5645.4     .05       0    5763      .1       0
Bank Sta=4995.1,5001.1
XS Rating Curve= 0 ,0
Exp/Cntr=0.3,0.1

Type RM Length L Ch R = 1 ,6712    ,532,532,532
BEGIN DESCRIPTION:
UNT 0085 IN HEWA 12.0
END DESCRIPTION:
XS GIS Cut Line= 3
      2638656.68     10077538.19      2637635.84      10077355.9
      2636766.04     10076934.02
#Sta/Elev= 30
  4305.1  2055.8  4628.3 2048.22  4707.4 2044.16  4810.1 2039.52  4927.9 2036.78
  4986.8 2033.44    4994 2030.96  5001.2 2030.13  5003.9 2029.63  5007.2 2030.13
  5014.4    2031  5024.5  2034.1  5036.5 2035.35  5105.8 2034.44  5135.9 2035.19
  5197.2 2036.35  5207.2 2036.33  5212.3 2035.45  5237.8 2036.65    5290 2037.21
  5325.1 2037.78  5394.7 2041.94  5588.2  2047.9  5747.9 2053.18  5828.2 2056.37
  6083.8    2063  6158.3 2066.11  6186.4  2066.3  6248.6 2068.94  6308.8 2070.39
#Mann= 9 ,-1 , 0
  4305.1     .16       0  4707.4      .1       0  5001.2     .07       0
  5007.2      .1       0  5036.5     .16       0  5135.9     .05       0
    5290      .1       0  5588.2     .05       0  5747.9      .1       0
Bank Sta=5001.2,5007.2
XS Rating Curve= 0 ,0
Exp/Cntr=0.3,0.1

Type RM Length L Ch R = 1 ,6180    ,442,442,442
BEGIN DESCRIPTION:
UNT 0085 IN HEWA 11.0
END DESCRIPTION:
XS GIS Cut Line= 3
      2639018.44     10077403.72      2637818.47     10076903.73
      2637418.44     10076903.73
#Sta/Elev= 30
    3722 2063.07  3798.8  2060.7  3866.6  2059.6  4121.2 2051.54  4144.5 2051.73
  4209.5 2049.36  4501.5 2043.22  4534.5 2042.51  4662.5  2035.3    4762 2033.64
  4853.5  2034.4  4913.6 2033.92  4930.4 2032.85  4935.8 2033.53  4954.3 2031.64
  4983.5 2030.93  4997.3 2027.49  5000.1 2026.99  5003.3 2027.49  5004.3 2027.55
  5012.8 2027.58  5019.3 2029.79  5024.5 2029.79    5032 2031.62    5072 2035.17
    5122 2035.85    5183 2038.78    5272 2044.28    5382 2048.39    5422 2050.76
#Mann= 8 ,-1 , 0
    3722     .16       0  3798.8      .1       0  4501.5     .16       0
  4662.5      .1       0  4997.3     .07       0  5003.3      .1       0
  5004.3     .05       0    5183      .1       0
Bank Sta=4997.3,5003.3
XS Rating Curve= 0 ,0
Exp/Cntr=0.3,0.1

Type RM Length L Ch R = 1 ,5738    ,420,420,420
BEGIN DESCRIPTION:
UNT 0085 IN HEWA 10.0
END DESCRIPTION:
XS GIS Cut Line= 3
      2639104.57     10077184.01      2637906.67     10076517.36
      2637162.64     10076444.51
#Sta/Elev= 30
  3560.9 2062.53  3762.5 2057.15  3888.3 2051.72  4087.2 2046.96    4109 2045.62
  4374.2 2040.25  4390.2  2040.7  4455.4 2037.79  4562.6 2036.23  4633.8 2033.58
  4699.3 2031.86  4744.1 2031.56  4807.6 2030.28    4851 2032.19  4970.2 2029.98
  4980.2  2029.1  4997.3 2024.47  5000.1 2023.97  5003.3 2024.47  5010.4 2025.22
  5017.9 2028.87  5038.4 2031.57  5060.6 2030.62  5208.4 2035.09  5271.6 2040.26
  5422.3 2046.64  5522.8 2053.35  5630.1  2054.8  5663.5 2055.53  5679.4 2056.93
#Mann= 10 ,-1 , 0
  3560.9      .1       0  4562.6     .16       0  4633.8      .1       0
  4699.3     .16       0  4744.1      .1       0  4997.3     .07       0
  5003.3      .1       0  5038.4     .05       0  5208.4      .1       0
  5630.1     .05       0
Bank Sta=4997.3,5003.3
XS Rating Curve= 0 ,0
Exp/Cntr=0.3,0.1

Type RM Length L Ch R = 1 ,5318    ,423,423,423
BEGIN DESCRIPTION:
UNT 0085 IN HEWA 9.0
END DESCRIPTION:
XS GIS Cut Line= 4
      2639125.43     10076996.53      2637807.72     10076038.19
      2637552.51     10075678.81      2637562.88     10075678.81
#Sta/Elev= 30
    3478 2066.73  3485.8 2062.63    3499 2059.26  3647.2 2054.31    3693 2053.95
  3710.9 2051.41  3749.4 2047.52  3985.9 2046.21  4000.5 2043.46  4029.9 2041.98
  4278.7 2035.28  4412.4 2035.49  4643.9    2033  4880.4 2027.93  4917.1 2025.37
  4949.5 2027.02  4973.5 2025.92  4992.1 2019.99  4994.9 2019.49  4998.1 2019.99
  5017.6 2026.88  5032.2 2028.77  5120.2 2027.53  5210.9 2026.25  5245.9 2028.53
  5315.9 2036.11  5375.8 2041.39  5440.3  2045.5  5482.1 2043.77  5558.5 2044.62
#Mann= 13 ,-1 , 0
    3478      .1       0  3647.2     .16       0  3710.9      .1       0
  4412.4     .05       0  4643.9     .16       0  4880.4      .1       0
  4949.5     .16       0  4992.1     .07       0  4998.1     .16       0
  5120.2     .05       0  5245.9      .1       0  5315.9     .05       0
  5375.8      .1       0
Bank Sta=4992.1,4998.1
XS Rating Curve= 0 ,0
Exp/Cntr=0.3,0.1

Type RM Length L Ch R = 1 ,4895    ,1054,1054,1054
BEGIN DESCRIPTION:
UNT 0085 IN HEWA 8.0
END DESCRIPTION:
XS GIS Cut Line= 2
      2639246.41     10076690.99      2637601.99      10075353.6
#Sta/Elev= 30
  3606.8 2058.44  3681.5 2055.62  3731.9 2047.96  4037.1 2046.88  4091.9 2044.24
  4105.7 2043.98    4328 2031.56  4377.5 2025.75  4455.8 2023.77  4502.9 2027.36
  4565.5 2026.44  4705.9 2025.91    4778 2026.19  4828.7 2025.16  4968.7 2023.67
  5000.9 2018.51  5003.6 2018.01  5006.9 2018.51    5047 2026.95  5074.3  2025.7
  5107.5 2023.26  5146.1 2022.85  5174.8 2030.91  5181.3 2036.82  5195.6 2039.46
  5272.3 2039.85  5444.9 2042.46  5549.5  2047.4  5636.6 2052.94  5726.4 2054.52
#Mann= 14 ,-1 , 0
  3606.8      .1       0  4091.9     .16       0  4105.7      .1       0
  4502.9     .16       0  4565.5     .12       0  4705.9     .16       0
    4778     .12       0  4828.7     .16       0  5000.9     .07       0
  5006.9     .16       0  5074.3      .1       0  5107.5     .16       0
  5272.3      .1       0  5549.5     .05       0
Bank Sta=5000.9,5006.9
XS Rating Curve= 0 ,0
Exp/Cntr=0.3,0.1

Type RM Length L Ch R = 1 ,3841    ,696,696,696
BEGIN DESCRIPTION:
UNT 0085 IN HEWA 7.0
END DESCRIPTION:
XS GIS Cut Line= 3
      2639380.96     10075827.18      2638977.31     10075603.22
      2638097.11     10075384.47
#Sta/Elev= 30
  4714.9 2041.68  4755.4 2040.92  4809.1 2036.94  4833.3 2034.19  4852.6  2031.2
  4858.3 2027.17  4866.4 2025.54  4880.1 2018.96  4889.3 2016.34  4901.8 2015.95
  4927.3 2018.55  4946.5 2020.05  4969.3 2019.59  4977.4 2018.21  4983.1  2015.1
  4993.5 2013.34  4996.1  2013.1  4998.9  2012.6  5002.1  2013.1  5036.9 2016.38
  5064.3 2021.06  5176.5 2021.74  5250.7 2023.48  5255.3 2023.57  5309.3 2025.67
  5540.5 2027.99  5697.5 2031.17  5771.7 2033.66  5972.5 2037.87  6083.5 2040.77
#Mann= 11 ,-1 , 0
  4714.9      .1       0  4833.3     .16       0  4927.3     .05       0
  4993.5      .1       0  4996.1     .07       0  5002.1      .1       0
  5250.7     .05       0  5255.3      .1       0  5540.5     .05       0
  5697.5      .1       0  5972.5     .05       0
Bank Sta=4996.1,5002.1
XS Rating Curve= 0 ,0
Exp/Cntr=0.3,0.1

Type RM Length L Ch R = 1 ,3145    ,275,275,275
BEGIN DESCRIPTION:
UNT 0085 IN HEWA 6.0
END DESCRIPTION:
XS GIS Cut Line= 2
       2639676.3     10074958.71      2638422.24     10075286.53
#Sta/Elev= 30
  4459.7 2037.77  4577.4 2035.27  4591.8 2036.17  4612.5 2034.66  4658.3 2034.51
  4698.7 2032.51  4705.5 2035.13  4715.9 2035.79    4820 2035.27  4824.3 2034.44
  4839.9 2031.44  4936.2 2027.42  4953.6 2024.56  4963.9 2020.43  4976.6 2011.76
  5002.3    2010    5005  2009.5  5008.3    2010  5024.6 2012.04  5057.5 2015.13
    5274 2017.59  5330.3 2019.79  5365.5 2022.69  5405.4 2023.57  5443.4 2024.85
  5546.6 2026.99  5648.6 2028.42  5690.6 2030.31    5753 2032.33  5755.9 2032.52
#Mann= 10 ,-1 , 0
  4459.7     .05       0  4824.3     .16       0  5002.3     .07       0
  5008.3     .16       0  5024.6      .1       0  5405.4     .05       0
  5443.4      .1       0  5546.6     .05       0  5690.6      .1       0
    5753     .05       0
Bank Sta=5002.3,5008.3
XS Rating Curve= 0 ,0
Exp/Cntr=0.3,0.1

Type RM Length L Ch R = 1 ,2870    ,334,334,334
BEGIN DESCRIPTION:
UNT 0085 IN HEWA 5.0
END DESCRIPTION:
XS GIS Cut Line= 3
      2639581.07     10074876.86      2639101.87     10074850.81
      2638377.91     10074991.44
#Sta/Elev= 30
    4411 2033.63  4461.7 2032.84  4483.7 2032.89    4561 2031.06    4684 2027.81
    4742 2022.33    4747 2023.92  4782.3 2020.51  4814.2    2019  4854.3 2015.75
  4890.1 2013.63  4958.2 2010.77  4962.7 2010.74  4965.4 2010.24  4968.7 2010.74
  5016.6    2011  5039.7 2013.42  5108.3  2014.2  5118.5 2015.96  5169.4 2016.65
  5194.8 2019.09    5200 2020.26  5220.4 2021.91  5262.4 2023.37  5349.8 2025.85
  5406.6 2026.54  5454.8 2027.88  5546.3 2031.77  5566.8 2031.66  5628.4 2033.31
#Mann= 9 ,-1 , 0
    4411     .16       0  4461.7     .05       0    4561     .16       0
  4782.3     .05       0  4958.2      .1       0  4962.7     .07       0
  4968.7      .1       0  5262.4     .08       0  5454.8     .05       0
Bank Sta=4962.7,4968.7
XS Rating Curve= 0 ,0
Exp/Cntr=0.3,0.1

Type RM Length L Ch R = 1 ,2536    ,105,105,105
BEGIN DESCRIPTION:
Mapping XS 7b4720fa
END DESCRIPTION:
XS GIS Cut Line= 2
      2639607.04     10074569.56      2638305.01      10074590.4
#Sta/Elev= 30
  4320.2 2033.42  4448.8 2028.34  4548.8 2025.43  4608.8 2021.82  4658.8 2019.82
  4778.8  2016.6  4888.6 2015.94  4893.6 2014.44  4918.9 2013.91  4928.9  2012.6
  4948.9 2007.93  4958.9 2007.31  4995.9  2007.2  4998.6  2006.7  5008.9 2008.12
 5027.28 2013.85  5028.9 2014.86  5038.9 2016.46  5048.9 2016.98  5098.9 2017.72
  5138.9 2019.46  5188.9 2020.28  5218.9 2021.31  5238.9 2022.97  5298.9  2024.9
  5338.9 2026.94  5438.9 2029.53  5478.9 2030.02  5528.9  2031.9  5622.4 2033.47
#Mann= 4 ,-1 , 0
  4320.2     .05       0  4918.9     .04       0 5027.28     .05       0
  5218.9      .1       0
Bank Sta=4918.9,5027.28
XS Rating Curve= 0 ,0
Exp/Cntr=0.3,0.1

Type RM Length L Ch R = 1 ,2431    ,334,334,334
BEGIN DESCRIPTION:
Mapping XS 770bfdd6
END DESCRIPTION:
XS GIS Cut Line= 2
      2639549.81     10074475.81      2638289.32     10074481.02
#Sta/Elev= 30
  4397.2 2030.98  4508.5 2028.04  4598.1 2024.33  4638.5 2023.27  4668.5 2021.42
  4698.5 2020.73  4718.5 2017.83  4828.5 2015.41  4858.5 2014.02  4878.5 2013.75
  4918.5  2014.1  4928.5 2013.55  4948.5 2011.56  4978.5 2007.28  4995.5 2006.13
  4998.3 2005.63  5018.5 2008.14  5038.5 2010.13  5048.5 2011.83  5058.5 2013.46
  5068.5 2014.53  5148.5 2017.69  5168.5 2017.46  5208.5 2018.78  5308.6  2023.9
  5368.6    2026  5428.6 2027.83  5524.4 2029.81  5548.6 2031.28  5657.7 2033.04
#Mann= 7 ,-1 , 0
  4397.2     .08       0  4598.1      .1       0  4878.5     .05       0
  4948.5     .04       0  5048.5     .05       0  5148.5     .08       0
  5524.4      .1       0
Bank Sta=4948.5,5048.5
XS Rating Curve= 0 ,0
Exp/Cntr=0.3,0.1

Type RM Length L Ch R = 1 ,2097    ,308,308,308
BEGIN DESCRIPTION:
UNT 0085 IN HEWA 4.0
END DESCRIPTION:
XS GIS Cut Line= 3
       2639508.1     10074366.43      2639101.87      10074152.9
       2638508.1      10074152.9
#Sta/Elev= 30
  4437.6 2028.98  4519.8 2026.02  4558.7 2024.88  4586.4 2023.51  4608.4 2023.39
    4717 2018.21  4779.1 2016.06  4795.5 2014.02  4832.6 2013.31  4839.6 2012.01
  4861.7 2010.37  4919.9 2009.22  4949.9 2007.76  4989.9 2004.26  4999.7  2002.6
  5019.9 2005.47  5039.9 2006.36  5049.9 2008.44  5059.9 2009.66  5128.6 2010.97
  5149.9 2011.51  5169.9 2013.04  5259.9 2014.82  5289.9 2016.04  5359.9  2021.3
  5389.9 2024.23  5419.9 2026.18  5442.6  2026.8  5459.9 2026.71  5490.3 2027.47
#Mann= 8 ,-1 , 0
  4437.6     .05       0  4519.8     .16       0    4717      .1       0
  4839.6     .05       0  4919.9     .04       0  5059.9     .05       0
  5128.6      .1       0  5442.6     .05       0
Bank Sta=4919.9,5059.9
XS Rating Curve= 0 ,0
Exp/Cntr=0.3,0.1

Type RM Length L Ch R = 1 ,1789    ,841,841,841
BEGIN DESCRIPTION:
UNT 0085 IN HEWA 3.0
END DESCRIPTION:
XS GIS Cut Line= 3
       2639677.5     10074251.73      2639068.13      10073855.9
      2638635.88     10073835.07
#Sta/Elev= 30
  4224.5 2030.11  4246.7 2029.59  4271.9 2029.35    4287  2028.2  4410.9 2024.34
  4440.3 2022.57  4479.5 2021.43  4497.6 2021.89  4525.6 2019.91  4620.1 2016.37
  4706.8 2013.71  4736.1 2014.25  4758.2 2013.06  4800.4 2012.81  4836.6 2010.69
  4851.8 2008.72  4912.2  2006.5  4938.8 2003.74  4970.8 2005.16  4997.9 2003.12
  5000.6 2002.62  5003.9 2003.12  5050.9 2008.42    5111 2008.27  5161.1 2011.28
  5201.1    2017  5261.2 2020.97    5307 2023.31    5312 2022.82  5383.9 2025.17
#Mann= 8 ,-1 , 0
  4224.5     .05       0  4246.7      .1       0  4440.3     .16       0
  4479.5      .1       0  4620.1     .05       0  4912.2      .1       0
  4997.9     .07       0  5003.9      .1       0
Bank Sta=4997.9,5003.9
XS Rating Curve= 0 ,0
Exp/Cntr=0.3,0.1

Type RM Length L Ch R = 1 ,1421    ,473,473,473
BEGIN DESCRIPTION:
Mapping XS c4cad072
END DESCRIPTION:
XS GIS Cut Line= 3
       2639763.5     10074010.36      2639082.11     10073476.53
      2638368.17     10073634.94
#Sta/Elev= 30
    4014 2028.06    4094 2024.59  4193.3 2021.67  4406.8 2014.12  4427.6 2017.87
  4450.2 2012.25  4485.5 2009.21  4514.4 2011.58  4520.7 2011.49  4535.2 2008.97
  4549.7 2009.12  4570.5 2007.91  4665.8 2007.07  4734.1 2007.21  4844.3 2004.97
  4914.1 2004.91  4973.6 2002.36    4993 1998.19  4995.8 1997.69    4999 1998.19
  5016.5 1999.59    5037 2006.04  5047.2 2007.37  5098.4 2008.56  5159.9 2013.63
  5190.6 2017.62  5209.5 2018.84  5355.5 2020.85  5476.7 2020.44  5610.9 2020.45
#Mann= 8 ,-1 , 0
    4014      .1       0  4193.3     .05       0  4665.8      .1       0
  4844.3     .16       0  4973.6      .1       0    4993     .07       0
    4999      .1       0  5476.7     .05       0
Bank Sta=4993,4999
XS Rating Curve= 0 ,0
Exp/Cntr=0.3,0.1
