--- WHITE OAK CREEK.prj (project) ---

Proj Title=WHITE OAK CREEK Base Level Engineering
Current Plan=p01
Default Exp/Contr=0.3,0.1
English Units
Geom File=g01
Flow File=f01
Plan File=p01
Y Axis Title=Elevation
X Axis Title(PF)=Main Channel Distance
X Axis Title(XS)=Station
BEGIN DESCRIPTION:
WHITE OAK CREEK
END DESCRIPTION:
DSS Export Rating Curves= 0
DSS Export Rating Curve Sorted= 0
DSS Export Volume Flow Curves= 0
DXF OffsetX= 0
DXF OffsetY= 0
DXF ScaleX= 1
DXF ScaleY= 10

--- WHITE OAK CREEK.p01 (plan) ---

Plan Title=Multiple Run
Short Identifier=Multiple
Geom File=g01
Flow File=f01
Subcritical Flow
K Sum by GR= 0
Std Step Tol= 0.01
Critical Tol= 0.01
Num of Std Step Trials= 20
Max Error Tol= 0.3
Flow Tol Ratio= 0.001
Split Flow NTrial= 30
Split Flow Tol= 0.02
Split Flow Ratio= 0.02
Log Output Level= 0
Friction Slope Method= 1
Unsteady Friction Slope Method= 2
Unsteady Bridges Friction Slope Method= 1
Parabolic Critical Depth
Global Vel Dist=  1 , 1 , 1
Global Log Level= 0
CheckData=True
Encroach Param= -1, 0, 0, 0
BEGIN DESCRIPTION:
Multiple Run
END DESCRIPTION:

--- WHITE OAK CREEK.f01 (steady flow) ---

Flow Title=Multiple
Program Version=4.10
Number of Profiles= 7
Profile Names=10-year,25-year,50-year,1pct_min,100-year,1pct_plu,500-year
River Rch & RM=WHITE OAK CREEK,Reach-1         ,68078
    1008    1450    1827    1678    2269    3068    3499
River Rch & RM=WHITE OAK CREEK,Reach-1         ,67736
    1486    2182    2786    2590    3502    4737    5535
River Rch & RM=WHITE OAK CREEK,Reach-1         ,63681
    1903    2827    3639    3407    4607    6231    7388
River Rch & RM=WHITE OAK CREEK,Reach-1         ,61450
    2428    3649    4734    4463    6036    8162    9816
River Rch & RM=WHITE OAK CREEK,Reach-1         ,58552
    2619    3947    5130    4843    6550    8858   10687
River Rch & RM=WHITE OAK CREEK,Reach-1         ,56702
    3263    4952    6466    6127    8286   11206   13620
River Rch & RM=WHITE OAK CREEK,Reach-1         ,49482
    4593    7058    9294    8872   11998   16226   20015
River Rch & RM=WHITE OAK CREEK,Reach-1         ,41998
    4695    7204    9478    9037   12222   16528   20341
River Rch & RM=WHITE OAK CREEK,Reach-1         ,38088
    5008    7701   10144    9684   13096   17711   21847
River Rch & RM=WHITE OAK CREEK,Reach-1         ,37243
    5008    7701   10144    9684   13096   17711   21847
River Rch & RM=WHITE OAK CREEK,Reach-1         ,36228
    6410    9926   13139   12595   17033   23035   28646
River Rch & RM=WHITE OAK CREEK,Reach-1         ,35249
    6410    9926   13139   12595   17033   23035   28646
River Rch & RM=WHITE OAK CREEK,Reach-1         ,29896
    7001   10866   14405   13827   18699   25288   31530
River Rch & RM=WHITE OAK CREEK,Reach-1         ,27762
    7001   10866   14405   13827   18699   25288   31530
River Rch & RM=WHITE OAK CREEK,Reach-1         ,25852
    7244   11255   14932   14341   19394   26228   32740
River Rch & RM=WHITE OAK CREEK,Reach-1         ,24422
    7294   11314   14994   14383   19452   26306   32759
River Rch & RM=WHITE OAK CREEK,Reach-1         ,17516
    8076   12568   16692   16043   21697   29343   36681
River Rch & RM=WHITE OAK CREEK,Reach-1         ,17021
    8076   12568   16692   16043   21697   29343   36681
River Rch & RM=WHITE OAK CREEK,Reach-1         ,15366
    8367   13014   17279   16600   22450   30360   37916
River Rch & RM=WHITE OAK CREEK,Reach-1         ,14169
    8367   13014   17279   16600   22450   30360   37916
River Rch & RM=WHITE OAK CREEK,Reach-1         ,7733
    8528   13262   17605   16910   22868   30927   38605
Boundary for River Rch & Prof#=WHITE OAK CREEK,Reach-1         , 1
Up Type= 0
Dn Type= 3
Dn Slope=0.009
Boundary for River Rch & Prof#=WHITE OAK CREEK,Reach-1         , 2
Up Type= 0
Dn Type= 3
Dn Slope=0.009
Boundary for River Rch & Prof#=WHITE OAK CREEK,Reach-1         , 3
Up Type= 0
Dn Type= 3
Dn Slope=0.009
Boundary for River Rch & Prof#=WHITE OAK CREEK,Reach-1         , 4
Up Type= 0
Dn Type= 3
Dn Slope=0.009
Boundary for River Rch & Prof#=WHITE OAK CREEK,Reach-1         , 5
Up Type= 0
Dn Type= 3
Dn Slope=0.009
Boundary for River Rch & Prof#=WHITE OAK CREEK,Reach-1         , 6
Up Type= 0
Dn Type= 3
Dn Slope=0.009
Boundary for River Rch & Prof#=WHITE OAK CREEK,Reach-1         , 7
Up Type= 0
Dn Type= 3
Dn Slope=0.009
DSS Import GetInterval= 0
DSS Import GetPeak= 0
DSS Import FillOption= 0

--- WHITE OAK CREEK.g01 (geometry) ---

Geom Title=Existing Conditions
Program Version=4.10

River Reach=WHITE OAK CREEK ,Reach-1
Reach XY= 30
      2662468.47     10030273.73      2667697.49     10028253.65
      2670220.81     10029559.47      2671856.06     10031394.66
      2671771.18     10032608.49      2673633.45     10033011.98
      2674051.58     10035472.57       2675075.9      10036024.8
      2675509.32     10037518.51      2677885.44     10036031.37
      2677867.79     10035270.41      2679726.05     10035976.66
      2680499.57      10034176.4      2682730.93      10034589.6
      2683226.97     10035663.51      2682439.65     10036962.33
      2683369.56       10037961.      2684582.97     10037632.39
      2684300.32     10039537.22      2687003.41     10041053.15
      2687820.39     10039320.97      2688660.93     10039329.65
      2689262.05     10041622.25      2692122.07     10044832.24
       2692279.5     10046003.98      2694397.98     10044904.71
      2694559.68     10048043.89      2696654.42     10049111.43
       2697461.4     10048769.93      2698446.82     10049953.35

Type RM Length L Ch R = 1 ,68078   ,342,342,342
BEGIN DESCRIPTION:
WHITE OAK CREEK 114.0
END DESCRIPTION:
XS GIS Cut Line= 2
      2662922.32     10030395.86      2662094.63     10029828.46
#Sta/Elev= 30
  4539.3 2073.98  4586.8 2072.23  4592.9 2071.32  4601.7  2071.6  4629.3 2069.77
  4688.4 2066.93  4715.4 2064.23  4846.8 2059.61  4931.9  2055.3  4960.5 2053.46
  4975.4 2050.99  4981.4 2049.05  4993.3 2047.96  4996.1 2047.46  4999.3 2047.96
  5004.7 2048.19  5026.1    2052  5041.1 2053.15  5068.1 2052.05  5162.3 2055.42
  5265.1 2060.92    5328  2064.7  5363.9  2068.7  5418.1 2072.84  5451.5 2075.59
  5471.5 2077.95  5501.3  2080.3  5507.4  2080.1  5513.9 2081.51  5542.8 2083.02
#Mann= 7 ,-1 , 0
  4539.3      .1       0  4629.3     .16       0  4993.3     .07       0
  4999.3     .16       0  5265.1      .1       0  5418.1     .16       0
  5451.5      .1       0
Bank Sta=4931.9,5162.3
XS Rating Curve= 0 ,0
Exp/Cntr=0.3,0.1

Type RM Length L Ch R = 1 ,67736   ,449,449,449
BEGIN DESCRIPTION:
Mapping XS e221245a
END DESCRIPTION:
XS GIS Cut Line= 2
      2663001.02     10030342.81      2662480.21     10029544.24
#Sta/Elev= 30
  4404.7 2071.53  4455.6 2068.54  4471.4  2066.8  4477.3 2066.98  4594.6    2060
  4637.3 2056.79  4702.1 2053.61  4709.7 2052.25  4715.7 2052.47  4724.9 2051.57
  4782.2 2050.23  4881.7  2050.9  4954.1 2050.04  4969.2  2048.7  4984.3 2046.02
  4990.3 2045.78  5002.4 2043.86  5005.2 2043.36  5008.4 2043.86  5012.5 2048.32
 5017.61  2051.7  5020.5 2054.02  5026.5 2056.33  5048.3 2062.26  5056.8 2063.83
    5108  2069.8    5120 2072.01  5140.8 2073.98  5222.7 2081.33  5358.1 2089.66
#Mann= 5 ,-1 , 0
  4404.7      .1       0  4455.6     .16       0  5002.4     .07       0
  5008.4     .16       0  5140.8      .1       0
Bank Sta=4724.9,5017.61
XS Rating Curve= 0 ,0
Exp/Cntr=0.3,0.1

Type RM Length L Ch R = 1 ,67287   ,455,455,455
BEGIN DESCRIPTION:
WHITE OAK CREEK 113.0
END DESCRIPTION:
XS GIS Cut Line= 3
      2663078.57     10030286.53      2663130.66     10029619.83
      2662882.03     10029402.28
#Sta/Elev= 30
  4517.6 2069.95  4542.5 2068.99  4560.5 2067.74  4590.6 2067.24  4660.8 2063.21
  4761.1 2054.43  4781.2 2050.57  4821.3 2047.59  4833.1  2047.3  4921.6 2045.41
  4931.7 2044.02  4971.8 2045.48  4981.8 2044.85  4991.8 2042.68  4998.9 2042.54
  5001.6 2042.04  5004.9 2042.54  5011.9 2042.91  5021.9 2045.28  5054.2 2045.62
  5072.1 2045.28  5090.6 2046.57  5095.6 2045.97  5112.2 2047.43  5186.3 2051.67
  5248.9  2056.6  5291.6 2061.64  5339.4 2064.98  5454.8 2075.71  5516.7 2079.81
#Mann= 7 ,-1 , 0
  4517.6      .1       0  4542.5     .16       0  4833.1      .1       0
  4998.9     .07       0  5004.9      .1       0  5054.2     .16       0
  5339.4      .1       0
Bank Sta=4821.3,5112.2
XS Rating Curve= 0 ,0
Exp/Cntr=0.3,0.1

Type RM Length L Ch R = 1 ,66832   ,436,436,436
BEGIN DESCRIPTION:
WHITE OAK CREEK 111.0
END DESCRIPTION:
XS GIS Cut Line= 3
      2663615.03     10030276.05      2663516.07     10029593.78
      2663074.81     10029297.88
#Sta/Elev= 30
  4427.5 2071.29  4551.1 2066.23    4577 2063.84  4582.1 2064.07    4642  2059.5
  4652.3  2057.8  4702.7 2054.06  4722.9 2051.26  4763.3 2049.08  4782.6 2046.37
  4787.6 2046.67  4813.8 2044.45  4852.8 2042.47  4857.8 2042.87  4874.4 2042.11
  4945.2 2041.71  4975.5 2038.64  4995.2 2038.04    4998 2037.54  5001.2 2038.04
  5015.9  2039.5  5036.1 2042.63  5116.9 2042.51    5165 2043.19  5235.8 2046.01
  5354.1 2051.41  5396.1 2054.63  5444.8 2057.19  5561.2 2065.84  5648.2 2069.96
#Mann= 5 ,-1 , 0
  4427.5      .1       0  4995.2     .07       0  5001.2      .1       0
  5235.8     .16       0  5444.8      .1       0
Bank Sta=4857.8,5036.1
XS Rating Curve= 0 ,0
Exp/Cntr=0.3,0.1

Type RM Length L Ch R = 1 ,66396   ,468,468,468
BEGIN DESCRIPTION:
WHITE OAK CREEK 110.0
END DESCRIPTION:
XS GIS Cut Line= 4
      2664052.53     10030197.94      2664057.74     10029895.87
      2663750.45     10029531.28      2663307.72     10029203.14
#Sta/Elev= 30
  4456.2 2060.01  4560.4 2054.69  4660.4 2051.42  4690.4 2049.15  4730.4 2048.93
  4756.9 2046.82  4766.3 2047.49  4780.6 2046.64  4794.9 2044.89  4801.4 2045.48
  4837.8 2043.28  4879.5 2042.65  4950.9 2037.19  4986.1 2032.61  4990.8 2030.76
  4993.6 2030.26  4996.8 2030.76  5008.1 2031.88  5014.7 2033.66    5029  2034.6
  5086.2 2035.03  5142.1 2037.12  5241.6 2037.72  5306.3 2041.22  5427.3 2042.75
  5509.1 2046.79  5531.5 2047.22  5592.2 2048.38  5677.8 2051.73  5786.2 2057.63
#Mann= 5 ,-1 , 0
  4456.2      .1       0  4990.8     .07       0  4996.8      .1       0
  5509.1     .16       0  5531.5      .1       0
Bank Sta=4950.9,5142.1
XS Rating Curve= 0 ,0
Exp/Cntr=0.3,0.1

Type RM Length L Ch R = 1 ,65928   ,470,470,470
BEGIN DESCRIPTION:
WHITE OAK CREEK 109.0
END DESCRIPTION:
XS GIS Cut Line= 2
      2664266.07     10030177.13      2664266.07     10029068.23
#Sta/Elev= 30
  4307.2 2054.69  4360.6 2053.36  4410.6 2051.39  4510.6 2046.44  4540.6 2044.44
  4610.6 2041.54  4640.6 2038.85  4720.6  2036.2  4748.7 2034.64  4800.6 2033.15
  4860.6 2030.37  4870.6 2030.28  4899.3  2031.4  4940.6  2032.1  4970.6  2028.1
  4982.8 2027.65  5007.6 2027.34  5010.3 2026.84  5013.6 2027.34  5020.6 2029.16
  5030.6  2033.5  5040.6 2037.69  5050.6 2040.65  5060.6 2042.85  5070.6 2043.95
  5160.6  2052.3  5299.3 2062.87  5320.6 2064.67  5357.9 2066.07  5416.1 2068.81
#Mann= 8 ,-1 , 0
  4307.2      .1       0  4748.7     .16       0  4899.3      .1       0
  4982.8     .16       0  5007.6     .07       0  5013.6     .16       0
  5299.3      .1       0  5357.9     .16       0
Bank Sta=4800.6,5030.6
XS Rating Curve= 0 ,0
Exp/Cntr=0.3,0.1

Type RM Length L Ch R = 1 ,65458   ,1018,1018,1018
BEGIN DESCRIPTION:
WHITE OAK CREEK 108.0
END DESCRIPTION:
XS GIS Cut Line= 4
      2664419.73     10030216.14      2664518.68     10029812.53
       2664716.6     10029671.91      2664625.44      10029132.8
#Sta/Elev= 30
  4461.7 2052.07  4520.1 2051.59    4598 2049.18  4686.5 2043.58  4733.2 2041.86
  4769.6 2038.36  4793.7 2037.77  4852.8 2033.56  4954.8 2028.28  4992.6 2024.18
  5005.2  2023.5  5011.9    2026    5020 2027.05  5070.4 2027.87  5076.6 2026.38
  5085.2 2026.95  5091.3 2024.54  5103.1 2022.88  5105.8 2022.38  5109.1 2022.88
  5112.2 2025.84  5118.1 2026.44  5172.1 2026.94  5198.4  2028.1  5201.6 2028.22
  5331.2 2036.39  5422.5 2040.66  5438.2 2042.68  5458.5 2043.61  5666.8 2050.17
#Mann= 7 ,-1 , 0
  4461.7     .16       0  4992.6      .1       0  5103.1     .07       0
  5109.1      .1       0  5172.1      .1       0  5198.4     .16       0
  5458.5      .1       0
Bank Sta=4954.8,5201.6
XS Rating Curve= 0 ,0
Exp/Cntr=0.3,0.1

Type RM Length L Ch R = 1 ,64440   ,196,196,196
BEGIN DESCRIPTION:
WHITE OAK CREEK 106.0
END DESCRIPTION:
XS GIS Cut Line= 4
      2665620.25     10030161.52      2665495.24     10029468.78
      2665044.72      10029229.2      2664698.37      10029104.2
#Sta/Elev= 30
  4170.1 2059.38  4452.4 2050.81  4635.3 2043.67  4662.2 2043.45  4696.2 2043.06
  4713.3 2040.79  4757.2 2038.33  4797.9 2037.99    4874 2034.39  4891.4 2033.25
    4927 2028.99  4941.2 2026.26    4963 2019.19  4972.3 2015.43    4985 2011.81
  4998.3 2010.32    5001 2009.82  5004.3 2010.32  5028.9 2016.28  5061.5 2018.18
  5177.1 2021.29  5233.5 2023.83  5297.6 2027.14  5357.4 2028.74  5472.4 2036.78
  5533.7 2038.84  5589.7 2043.03  5622.3 2043.56  5699.2 2044.91  5752.5 2048.58
#Mann= 7 ,-1 , 0
  4170.1      .1       0  4662.2     .16       0  4941.2      .1       0
  4998.3     .07       0  5004.3      .1       0  5233.5     .16       0
  5622.3      .1       0
Bank Sta=4963,5061.5
XS Rating Curve= 0 ,0
Exp/Cntr=0.3,0.1

Type RM Length L Ch R = 1 ,64244   ,563,563,563
BEGIN DESCRIPTION:
WHITE OAK CREEK 105.0
END DESCRIPTION:
XS GIS Cut Line= 3
      2666013.44     10029648.45      2665128.05      10028976.6
       2664962.4      10028821.3
#Sta/Elev= 30
  4309.7 2046.39  4438.4 2042.45    4480 2038.25  4544.5 2035.37  4599.8 2031.11
  4643.6 2029.57  4698.6 2027.39  4730.2 2029.09  4744.2 2027.95  4787.8 2028.67
    4931 2021.31  4937.6 2020.99  4958.4 2016.36  4966.7 2012.83  4999.1 2009.44
  5001.8 2008.94  5005.1 2009.44  5016.6 2013.19  5037.4 2016.64    5044 2017.48
    5052    2016  5072.8 2016.11    5130 2018.97    5208 2022.13  5316.1 2030.03
  5357.9 2034.91  5444.2 2038.39  5479.4 2041.64  5562.5  2045.2  5648.2 2049.18
#Mann= 9 ,-1 , 0
  4309.7      .1       0  4599.8     .16       0  4643.6      .1       0
  4698.6     .16       0    4931      .1       0  4999.1     .07       0
  5005.1      .1       0    5130     .16       0  5562.5      .1       0
Bank Sta=4958.4,5037.4
XS Rating Curve= 0 ,0
Exp/Cntr=0.3,0.1

Type RM Length L Ch R = 1 ,63681   ,751,751,751
BEGIN DESCRIPTION:
WHITE OAK CREEK 103.0
END DESCRIPTION:
XS GIS Cut Line= 3
      2666263.47     10029335.97       2665654.1     10028643.26
      2665253.27     10028440.25
#Sta/Elev= 30
  4312.8  2038.9  4417.2 2031.11  4459.9 2029.61  4526.6 2024.73  4587.1 2021.84
  4615.5 2019.08  4721.8 2020.26  4792.9 2015.21  4891.6 2012.23  4955.2 2010.65
  4991.2 2007.33  5019.7 2007.26  5040.6 2008.81  5058.6 2007.07  5061.4 2006.57
  5064.6 2007.07 5078.18 2012.39  5082.2 2015.07  5097.5 2020.51  5111.7  2023.8
    5126 2025.39    5182 2029.81  5235.4 2031.49  5275.3 2037.14  5360.4 2040.32
  5441.2 2045.03  5513.7 2046.55  5580.5 2050.65  5647.3 2051.32  5684.7 2053.24
#Mann= 6 ,-1 , 0
  4312.8     .16       0  4526.6      .1       0  5058.6     .07       0
  5064.6      .1       0  5082.2     .16       0  5360.4      .1       0
Bank Sta=4891.6,5078.18
XS Rating Curve= 0 ,0
Exp/Cntr=0.3,0.1

Type RM Length L Ch R = 1 ,62930   ,356,356,356
BEGIN DESCRIPTION:
WHITE OAK CREEK 102.0
END DESCRIPTION:
XS GIS Cut Line= 3
      2666560.34     10029184.88      2666450.97     10028398.47
      2666253.29     10028153.97
#Sta/Elev= 30
    4361 2041.85  4422.7 2039.53  4493.4  2034.4  4574.2 2030.48  4634.8 2026.18
  4725.6 2022.48  4745.8 2020.74  4772.5 2015.62  4836.7 2006.22    4867 2002.84
  4937.6 2004.79  4967.9 2004.75  4992.4 2002.75  4995.2 2001.66    4998 2001.16
  5001.2 2001.66    5026 2003.53  5048.7 2004.45  5069.1 2002.62  5099.2 2001.74
  5140.7 2005.98  5154.8 2009.77  5163.4 2010.22  5173.9 2012.04  5231.2 2015.29
  5259.9 2020.38  5309.5 2022.79  5330.3  2024.8  5387.9 2027.21  5469.4 2032.75
#Mann= 5 ,-1 , 0
    4361     .16       0  4995.2     .07       0  5001.2     .16       0
    5026      .1       0  5163.4     .16       0
Bank Sta=4836.7,5140.7
XS Rating Curve= 0 ,0
Exp/Cntr=0.3,0.1

Type RM Length L Ch R = 1 ,62574   ,288,288,288
BEGIN DESCRIPTION:
WHITE OAK CREEK 101.0
END DESCRIPTION:
XS GIS Cut Line= 3
      2666872.85     10029070.37      2666805.14     10028362.01
      2666453.77     10028098.49
#Sta/Elev= 30
  4419.3 2040.09  4519.6 2035.27  4556.6 2032.46  4677.1  2025.6  4717.3 2024.63
  4777.6 2021.26    4833 2015.51  4898.1  2011.4  4928.3 2006.61  4935.8 2003.37
  4948.3 1999.91  4958.4 1999.35  4978.5 1999.83  4995.6 1998.45  4998.3 1997.95
  5001.6 1998.45  5038.5 2000.95  5078.9 2002.27  5149.3 2001.28  5176.7 2002.29
  5234.7 2001.47  5290.9 2002.78  5305.5 2004.06  5326.7 2008.09  5355.5 2012.09
  5370.1 2013.56  5384.7 2013.95  5390.9 2015.11  5440.9 2020.35  5570.1 2025.98
#Mann= 3 ,-1 , 0
  4419.3     .16       0  4995.6     .07       0  5001.6     .16       0
Bank Sta=4935.8,5305.5
XS Rating Curve= 0 ,0
Exp/Cntr=0.3,0.1

Type RM Length L Ch R = 1 ,62286   ,836,836,836
BEGIN DESCRIPTION:
WHITE OAK CREEK 100.0
END DESCRIPTION:
XS GIS Cut Line= 4
      2667128.06      10029065.1      2667190.55     10028591.18
      2666919.72     10028122.43       2666623.2     10027935.15
#Sta/Elev= 30
  4305.3 2035.06  4326.9 2034.22  4357.1 2031.52  4454.1 2028.08  4575.1 2023.68
  4653.6  2022.1    4690 2018.35  4745.1  2014.8  4813.4 2011.28  4819.1 2011.75
  4834.9 2010.01  4849.7  2009.9  4872.2 2008.16  4921.1 2006.72  4958.4 2002.78
    4960 2001.95  4974.2 1998.33  4992.7 1996.03  4995.5 1995.53  4998.7 1996.03
  5054.6 1999.02  5103.8 2000.14  5149.9 1999.45  5199.6 2000.29  5258.4  1999.8
    5426 2002.02  5483.6 2006.82  5514.2 2010.46  5614.2 2014.48  5675.4  2020.1
#Mann= 5 ,-1 , 0
  4305.3     .16       0  4454.1      .1       0  4745.1     .16       0
  4992.7     .07       0  4998.7     .16       0
Bank Sta=4960,5426
XS Rating Curve= 0 ,0
Exp/Cntr=0.3,0.1

Type RM Length L Ch R = 1 ,61450   ,504,504,504
BEGIN DESCRIPTION:
WHITE OAK CREEK 99.0
END DESCRIPTION:
XS GIS Cut Line= 2
      2667284.29     10029112.03      2668075.97     10028039.09
#Sta/Elev= 30
  4038.4 2033.04    4069 2030.68  4146.9 2027.61  4284.1    2023  4352.3 2018.95
    4376 2016.78  4555.6 2007.43  4583.1 2004.04  4632.8 2000.62    4691 1998.69
  4806.2 1997.12  4856.3 1995.44  4883.4 1993.71  4912.6 1993.96    4969 1992.46
  4977.4  1991.7  4995.2 1986.04    4998 1985.54  5001.2 1986.04  5005.6 1986.38
  5019.2  1989.7  5042.1 1990.65 5053.98 1995.86  5083.8 2014.02  5105.1 2023.26
  5184.1 2039.04    5228 2042.04    5255 2044.73  5305.2 2046.09  5371.8  2049.3
#Mann= 7 ,-1 , 0
  4038.4     .16       0  4146.9      .1       0  4352.3     .16       0
    4691      .1       0  4995.2     .07       0  5001.2      .1       0
  5019.2     .16       0
Bank Sta=4856.3,5053.98
XS Rating Curve= 0 ,0
Exp/Cntr=0.3,0.1

Type RM Length L Ch R = 1 ,60946   ,549,549,549
BEGIN DESCRIPTION:
WHITE OAK CREEK 98.0
END DESCRIPTION:
XS GIS Cut Line= 2
       2667409.3     10029429.72      2668543.53     10028378.74
#Sta/Elev= 30
  3886.8 2033.58  3918.7 2033.35  3975.4 2029.68  4088.8 2025.69  4244.1 2023.62
  4265.7 2020.77    4294 2018.16    4315 2017.66  4329.2  2015.6  4428.4 2010.85
  4463.6 2010.26  4548.6 2002.59  4633.6 1998.87  4684.7 1999.09  4774.8 1996.52
    4853 1991.95  4888.2 1987.51  4915.8 1989.16  4951.7 1989.15  4998.6 1982.38
  5001.3 1981.88  5004.6 1982.38  5015.8 1984.45  5029.9 1992.26  5071.9 2006.53
    5136 2021.31  5199.5 2026.46  5298.7 2031.14    5348 2035.74  5433.1 2038.58
#Mann= 5 ,-1 , 0
  3886.8     .16       0  4684.7      .1       0  4915.8     .16       0
  4998.6     .07       0  5004.6     .16       0
Bank Sta=4853,5029.9
XS Rating Curve= 0 ,0
Exp/Cntr=0.3,0.1

Type RM Length L Ch R = 1 ,60397   ,582,582,582
BEGIN DESCRIPTION:
WHITE OAK CREEK 96.0
END DESCRIPTION:
XS GIS Cut Line= 3
      2667919.71     10029710.98      2668768.68     10028898.47
      2668924.93     10028492.21
#Sta/Elev= 30
  4069.5 2039.43  4116.2 2035.46  4201.1 2034.43  4307.1 2027.77  4448.6 2022.68
  4540.4 2014.37  4632.6 2009.58    4682 2002.17  4752.7 1996.38  4827.2 1992.87
  4908.4  1987.9  4943.6 1987.08  4984.1 1981.24  4997.2 1978.77    5000 1978.27
  5003.2 1978.77  5035.8 1984.25  5064.1 1982.94  5106.2 1985.57  5134.5 1984.23
  5184.2 1985.76  5205.3 1988.52  5240.8 1993.61  5244.4 1995.52  5249.8 1995.52
  5256.5 1997.95  5292.6 2005.49  5395.8 2018.53  5589.7 2024.86  5679.9 2025.43
#Mann= 5 ,-1 , 0
  4069.5     .16       0  4827.2      .1       0  4984.1     .16       0
  4997.2     .07       0  5003.2     .16       0
Bank Sta=4908.4,5205.3
XS Rating Curve= 0 ,0
Exp/Cntr=0.3,0.1

Type RM Length L Ch R = 1 ,59815   ,560,560,560
BEGIN DESCRIPTION:
WHITE OAK CREEK 95.0
END DESCRIPTION:
XS GIS Cut Line= 4
      2668674.92     10029893.27      2668977.01     10029622.43
      2669128.05     10029091.18      2669055.14      10028513.1
#Sta/Elev= 30
  4390.1 2032.34  4456.1 2028.15  4597.3 2023.19  4668.4 2016.49  4804.9 2008.25
    4859 1999.58  4919.2  1995.5  4960.7 1987.29  4965.9 1988.49 4969.09 1984.37
  4971.2 1981.59  4981.6 1977.05    4992    1974  5001.9 1973.59  5004.7 1973.09
  5007.9 1973.59  5033.6 1976.76  5038.8  1979.5  5072.7 1979.98    5096 1983.14
  5111.8 1983.22  5137.6 1978.58  5158.4 1981.15  5199.9 1982.93  5382.8 1984.25
  5463.1 1994.89  5567.3 2005.49  5668.1 2010.61  5748.7 2016.86  5930.8 2020.74
#Mann= 3 ,-1 , 0
  4390.1     .16       0  5001.9     .07       0  5007.9     .16       0
Bank Sta=4969.09,5382.8
XS Rating Curve= 0 ,0
Exp/Cntr=0.3,0.1

Type RM Length L Ch R = 1 ,59255   ,703,703,703
BEGIN DESCRIPTION:
WHITE OAK CREEK 93.0
END DESCRIPTION:
XS GIS Cut Line= 4
       2669409.3     10030179.75      2669575.97      10029606.8
      2669602.01     10029325.55      2669154.08     10028554.69
#Sta/Elev= 30
  4279.5 2008.77  4314.8  2006.4    4365 2002.08  4431.6 1998.67    4543 1997.96
  4858.6 1990.33  4919.1 1985.73  4951.7 1978.39  4961.1 1976.35  4969.7 1972.74
  4996.8 1971.18  4999.5 1970.68  5002.8 1971.18  5019.9 1974.04  5065.5 1978.51
  5110.3 1979.59  5130.3 1977.82  5162.6 1977.59  5257.2 1979.84  5322.7 1979.06
  5374.7 1980.59  5542.4 1981.86  5565.6 1983.39  5600.3 1989.18  5674.3 1994.67
  5770.4 1999.06  5834.9 2006.15  5930.9  2010.7  5995.5 2016.25  6050.2 2017.82
#Mann= 5 ,-1 , 0
  4279.5     .16       0  4314.8      .1       0  4919.1     .16       0
  4996.8     .07       0  5002.8     .16       0
Bank Sta=4951.7,5065.5
XS Rating Curve= 0 ,0
Exp/Cntr=0.3,0.1

Type RM Length L Ch R = 1 ,58552   ,497,497,497
BEGIN DESCRIPTION:
WHITE OAK CREEK 92.0
END DESCRIPTION:
XS GIS Cut Line= 3
      2669523.93     10030200.53      2670117.64     10029783.89
      2670549.93     10028950.55
#Sta/Elev= 30
  4029.8 2006.55  4071.9 2001.58  4138.3 1997.71  4194.9 1997.53  4403.2 1989.64
  4605.4 1978.78  4800.3 1974.58  4845.4 1973.54  4902.7 1969.04    4947 1969.03
  4982.6 1966.17  4985.3 1965.67  4988.6 1966.17  5007.7  1966.5  5024.5 1969.37
  5059.5 1974.77  5068.4 1976.24  5074.1 1979.62  5090.6 1983.91  5096.2  1987.8
  5134.8 1997.61  5140.4 2000.82  5156.9 2004.24  5162.6 2007.57  5179.1 2011.78
  5184.7 2014.97  5228.9 2026.08  5363.6 2034.17    5533 2039.23  5693.9 2041.12
#Mann= 5 ,-1 , 0
  4029.8     .16       0  4071.9      .1       0  4982.6     .07       0
  4988.6      .1       0  5024.5     .16       0
Bank Sta=4800.3,5059.5
XS Rating Curve= 0 ,0
Exp/Cntr=0.3,0.1

Type RM Length L Ch R = 1 ,58055   ,433,433,433
BEGIN DESCRIPTION:
WHITE OAK CREEK 91.0
END DESCRIPTION:
XS GIS Cut Line= 3
      2669742.63     10030304.72      2670617.64     10029924.51
      2670872.78     10029018.49
#Sta/Elev= 30
  4225.4 1998.87  4234.8 1998.78  4314.6 1997.34  4449.8 1990.99  4641.3 1975.36
  4787.4 1973.02  4798.7 1971.52  4839.8 1972.28  4853.2 1970.58    4921 1972.12
  4962.3 1966.64  5002.9 1966.12  5005.6 1965.62  5008.9 1966.12  5038.3 1966.78
  5060.4 1970.97  5067.2 1974.33  5096.1 1982.39  5143.5 1990.79  5276.8  1992.3
  5310.9 1995.42  5423.3 1999.72  5457.4 2004.72  5491.4 2008.03  5496.6 2007.18
  5523.1 2011.41  5716.4 2025.59  5956.1 2026.76  6087.8 2026.38  6120.7 2027.93
#Mann= 6 ,-1 , 0
  4225.4     .16       0  4234.8      .1       0  5002.9     .07       0
  5008.9      .1       0  5143.5     .16       0  5956.1      .1       0
#XS Ineff= 1 ,-1
 4754.26 4914.77 1972.62
Permanent Ineff=
       F
Bank Sta=4921,5060.4
XS Rating Curve= 0 ,0
Exp/Cntr=0.3,0.1

Type RM Length L Ch R = 1 ,57622   ,415,415,415
BEGIN DESCRIPTION:
WHITE OAK CREEK 90.0
END DESCRIPTION:
XS GIS Cut Line= 3
      2669898.91     10030539.09      2671023.89     10030304.72
      2671392.81     10030138.44
#Sta/Elev= 30
  4253.6 2003.06  4301.8 1998.21  4352.9 1997.51  4357.2 1997.56  4416.6 1996.08
  4518.7 1990.15  4590.2 1981.43  4620.9 1975.42  4652.1 1971.97  4830.5 1969.83
  4917.1 1966.69  4978.4 1961.68  5016.3 1961.45    5019 1960.95  5022.3 1961.45
  5042.3 1965.93  5049.9  1970.1  5087.3 1974.48  5223.5 1977.96  5304.8 1982.21
  5346.1 1984.96  5402.5 1991.79  5495.7 1999.88  5513.3 2003.43  5518.8 2002.89
  5536.4 2006.94  5611.3 2016.96  5714.9 2025.01  5778.3 2027.69  5807.4 2028.13
#Mann= 8 ,-1 , 0
  4253.6     .16       0  4352.9      .1       0  4357.2     .16       0
  4830.5      .1       0  5016.3     .07       0  5022.3      .1       0
  5304.8     .16       0  5778.3      .1       0
Bank Sta=4917.1,5042.3
XS Rating Curve= 0 ,0
Exp/Cntr=0.3,0.1

Type RM Length L Ch R = 1 ,57207   ,505,505,505
BEGIN DESCRIPTION:
WHITE OAK CREEK 89.0
END DESCRIPTION:
XS GIS Cut Line= 4
      2670029.14     10030820.35      2670393.68     10030841.18
      2670883.26     10030757.85      2671383.29     10030335.95
#Sta/Elev= 30
  4314.6 1999.48  4454.2 1997.33  4534.3 1993.23  4644.5 1990.83  4704.9 1987.92
  4745.5  1983.8  4826.6 1969.35  4894.6 1966.71  4948.3 1964.86  4968.6 1960.09
  4988.1 1953.92  4996.1 1953.57  4998.8 1953.07  5002.1 1953.57  5029.5 1955.68
  5053.4 1956.01  5085.5 1960.95  5100.5 1962.41  5113.6  1965.1  5141.5 1966.89
  5204.4  1966.2  5339.6 1968.62  5403.3 1972.92  5447.6  1979.5  5565.9 2000.76
  5608.8 2012.21  5651.7 2020.24  5729.7 2026.33  5793.6 2028.53  5830.6 2029.07
#Mann= 8 ,-1 , 0
  4314.6     .16       0  4894.6      .1       0  4996.1     .07       0
  5002.1      .1       0  5085.5     .16       0  5141.5      .1       0
  5447.6     .16       0  5793.6      .1       0
Bank Sta=4948.3,5113.6
XS Rating Curve= 0 ,0
Exp/Cntr=0.3,0.1

Type RM Length L Ch R = 1 ,56702   ,365,365,365
BEGIN DESCRIPTION:
WHITE OAK CREEK 88.0
END DESCRIPTION:
XS GIS Cut Line= 4
      2670549.96     10031851.56      2671049.93     10031346.39
      2671065.55     10030763.05      2671523.02     10030378.37
#Sta/Elev= 30
  4012.8 2003.93  4165.7  1993.9  4455.7 1982.55  4540.6 1974.08  4696.1 1974.06
  4756.2 1973.46  4786.2 1971.23  4886.3 1971.11  4926.3  1969.5  4936.3 1967.98
 4951.14 1962.78  4966.3 1955.75  4983.3 1953.81  4986.1 1953.31  4989.3 1953.81
  4990.3 1953.82  5046.3 1956.13  5086.3 1962.99  5099.7 1963.82  5358.5 1966.17
  5401.4 1969.17    5439 1976.51  5493.8 1987.39  5599.2    2015  5621.3 2019.23
  5663.7 2024.51  5745.6 2024.65  5849.4  2027.5  5890.9 2028.93  5904.8 2029.39
#Mann= 9 ,-1 , 0
  4012.8      .1       0  4983.3     .07       0  4989.3      .1       0
  4990.3     .16       0  5099.7      .1       0    5439     .16       0
  5745.6      .1       0  5849.4     .16       0  5890.9      .1       0
Bank Sta=4951.14,5086.3
XS Rating Curve= 0 ,0
Exp/Cntr=0.3,0.1

Type RM Length L Ch R = 1 ,56337   ,412,412,412
BEGIN DESCRIPTION:
WHITE OAK CREEK 87.0
END DESCRIPTION:
XS GIS Cut Line= 3
      2670601.98     10031851.62      2671315.55     10031377.64
      2671726.79     10030378.19
#Sta/Elev= 30
  3884.9 2002.17    3922 2000.66  4024.7 1993.95  4125.9 1990.54  4183.1 1986.22
  4270.3 1982.53  4378.5 1973.54  4467.8 1971.57  4558.9 1969.43  4667.1 1962.78
  4692.2 1963.05  4832.3 1961.45    4908 1962.68  4940.4 1958.32    4959 1953.49
  4961.8 1952.99    4965 1953.49  5037.7 1953.55  5070.2 1958.73  5076.7 1959.94
  5221.6 1961.56    5254  1963.5  5275.6 1967.36  5300.2 1976.96  5337.8 1993.59
    5373 1999.58  5473.8 2005.67  5521.7 2011.86  5802.6 2031.09  5822.3 2033.15
#Mann= 8 ,-1 , 0
  3884.9     .16       0    3922      .1       0  4467.8     .05       0
  4692.2      .1       0    4959     .07       0    4965      .1       0
  5300.2     .16       0  5802.6      .1       0
Bank Sta=4940.4,5070.2
XS Rating Curve= 0 ,0
Exp/Cntr=0.3,0.1

Type RM Length L Ch R = 1 ,55925   ,829,829,829
BEGIN DESCRIPTION:
WHITE OAK CREEK 86.0
END DESCRIPTION:
XS GIS Cut Line= 3
      2670596.76     10032049.54      2671612.43     10031466.18
      2672200.97     10030908.89
#Sta/Elev= 30
  3603.3 2013.39  3645.3 2011.85  3732.1 2003.56  3797.4 2000.16  4101.1 1982.07
  4165.8 1973.11  4246.4 1970.18  4343.9 1963.29  4423.2 1959.51  4504.1 1958.09
  4729.5 1959.53  4801.7  1959.1  4823.2 1956.82  4943.3 1952.54    4997 1946.73
  4999.7 1946.23    5003 1946.73    5021  1948.7  5042.4 1957.18  5056.6 1958.36
  5127.7 1955.71  5155.3 1959.41  5190.9 1974.46  5197.8  1975.6  5219.2 1985.62
  5240.3 1992.05  5247.5 1996.09  5304.2 2010.94  5410.2 2020.13  5585.1 2025.61
#Mann= 7 ,-1 , 0
  3603.3     .16       0  3797.4      .1       0  4343.9     .05       0
  4504.1      .1       0    4997     .07       0    5003      .1       0
  5127.7     .16       0
Bank Sta=4823.2,5042.4
XS Rating Curve= 0 ,0
Exp/Cntr=0.3,0.1

Type RM Length L Ch R = 1 ,55096   ,564,564,564
BEGIN DESCRIPTION:
WHITE OAK CREEK 85.0
END DESCRIPTION:
XS GIS Cut Line= 4
      2670549.93     10032221.39      2671414.51     10031971.39
      2671956.18     10032138.05      2672336.12     10031378.17
#Sta/Elev= 30
  3803.2 2016.95  3853.9 2014.38  3921.1 2011.15  4002.6 2002.23  4210.8 1991.87
  4316.9 1984.49  4500.5 1966.34    4530 1961.69  4567.8 1958.57  4664.5 1956.15
  4861.6 1952.44  4894.3  1951.5  4961.9 1943.81  4964.7 1943.31  4967.9 1943.81
  5010.8  1945.1  5030.3 1953.82  5035.6  1953.2  5042.1 1955.35  5100.9 1961.28
    5199  1963.9  5242.2 1962.39  5333.6 1970.44  5359.6 1971.02  5517.3 1977.26
  5611.5 1981.84  5842.3 1997.83  5954.1 2008.64  6021.2 2017.51  6119.5 2023.87
#Mann= 10 ,-1 , 0
  3803.2      .1       0  3853.9     .16       0  4002.6      .1       0
    4530     .05       0  4664.5      .1       0  4961.9     .07       0
  4967.9      .1       0  5359.6     .16       0  5517.3      .1       0
  5611.5     .16       0
Bank Sta=4861.6,5030.3
XS Rating Curve= 0 ,0
Exp/Cntr=0.3,0.1

Type RM Length L Ch R = 1 ,54532   ,704,704,704
BEGIN DESCRIPTION:
WHITE OAK CREEK 83.0
END DESCRIPTION:
XS GIS Cut Line= 3
      2671075.95     10033148.49      2672190.55     10032153.68
      2672393.47     10031388.83
#Sta/Elev= 30
  4118.6 2025.76  4357.5  2023.9    4513 2019.28  4591.1 2014.04  4661.9 2003.65
  4711.7 1999.98  4742.2 1995.35  4775.5    1991    4804 1984.39  4839.1 1972.92
    4860  1964.1  4888.4 1956.94  4945.3 1951.39  4959.5  1947.9  4973.7 1941.91
  5011.6 1941.67  5013.3 1941.62  5016.1 1941.12  5019.3 1941.62  5073.2 1947.72
  5203.8 1951.55  5341.4 1951.15  5420.1 1952.45  5512.8 1961.31  5645.6 1970.47
  5821.9 1979.52  5856.8 1983.71  6150.5 2004.73  6248.3 2017.69  6403.9 2024.26
#Mann= 10 ,-1 , 0
  4118.6      .1       0  4742.2     .05       0  5011.6      .1       0
  5013.3    .035       0  5019.3      .1       0  5203.8     .05       0
  5341.4      .1       0  5512.8     .16       0  5645.6      .1       0
  5821.9     .16       0
Bank Sta=4959.5,5073.2
XS Rating Curve= 0 ,0
Exp/Cntr=0.3,0.1

Type RM Length L Ch R = 1 ,53828   ,565,565,565
BEGIN DESCRIPTION:
WHITE OAK CREEK 82.0
END DESCRIPTION:
XS GIS Cut Line= 4
      2671742.67     10033403.66      2672367.64      10033044.3
      2672362.43     10032570.35       2672529.1     10031361.99
#Sta/Elev= 30
  4013.8 2006.93  4165.5 1998.22    4232 1995.02  4299.8 1992.39  4365.6 1987.57
  4482.4 1982.62  4551.1    1976  4707.6 1970.89  4825.3 1966.38  4895.3 1959.36
  4935.3 1953.63  4965.3  1940.5  4975.3 1932.45  5002.3 1931.49  5005.1 1930.99
  5008.3 1931.49  5045.3 1939.81  5075.3 1941.35  5105.3 1945.06  5225.5 1948.18
  5439.2 1949.11  5500.3 1955.96  5588.9 1969.53  5721.4 1977.23  5745.9 1980.29
  5912.9 1995.11  6053.2 2004.31  6200.1 2018.01  6235.1 2019.03  6428.5 2021.91
#Mann= 15 ,-1 , 0
  4013.8      .1       0  4165.5     .16       0    4232      .1       0
  4299.8     .16       0  4365.6      .1       0  4482.4     .16       0
  4707.6      .1       0  5002.3     .07       0  5008.3      .1       0
  5500.3     .16       0  5721.4      .1       0  5745.9     .16       0
  5912.9      .1       0  6200.1     .16       0  6235.1      .1       0
Bank Sta=4965.3,5075.3
XS Rating Curve= 0 ,0
Exp/Cntr=0.3,0.1

Type RM Length L Ch R = 1 ,53263   ,625,625,625
BEGIN DESCRIPTION:
WHITE OAK CREEK 80.0
END DESCRIPTION:
XS GIS Cut Line= 4
      2672555.16      10033554.7      2672940.55     10033122.43
      2672893.68     10031997.43      2672503.26     10030805.34
#Sta/Elev= 30
  4019.9 1989.66  4065.3  1987.8    4143 1981.32  4228.3 1976.26  4440.7 1967.25
  4647.8 1956.48  4722.4 1951.03    4928 1939.39  4947.2 1936.03    4968 1935.38
  4978.1 1930.07  5015.1 1929.46  5017.8 1928.96  5021.1 1929.46  5068.1 1932.58
  5078.1 1934.49  5088.1 1939.18  5118.2 1943.46  5388.4 1948.45  5439.8 1954.72
  5538.5 1970.51  5617.4 1975.82  5825.5  1988.8  6011.3 1995.31  6080.3 2000.49
    6177 2003.09  6384.1  2014.8  6595.1  2019.8  6701.8 2020.56  6979.4 2023.37
#Mann= 10 ,-1 , 0
  4019.9      .1       0  4722.4     .16       0  4947.2      .1       0
  5015.1     .07       0  5021.1      .1       0  5439.8     .16       0
  5617.4      .1       0    6177     .16       0  6384.1      .1       0
  6701.8     .16       0
Bank Sta=4928,5088.1
XS Rating Curve= 0 ,0
Exp/Cntr=0.3,0.1

Type RM Length L Ch R = 1 ,52638   ,491,491,491
BEGIN DESCRIPTION:
WHITE OAK CREEK 79.0
END DESCRIPTION:
XS GIS Cut Line= 3
      2672831.15     10033565.17      2673810.35     10032533.89
      2673924.93     10031502.64
#Sta/Elev= 30
  4030.6 1981.62  4180.9  1971.3  4254.3 1965.94  4317.4 1961.43  4384.6 1957.17
  4467.6  1952.7    4654 1944.42  4680.5 1943.83  4751.1 1938.93  4826.5 1939.93
  4871.6 1938.93  4906.8 1935.34  4974.6 1927.24  4977.3 1926.74  4980.6 1927.24
    5020 1927.83  5055.2 1934.46  5119.1 1941.49  5232.3 1944.75  5253.4 1949.06
    5296 1962.97  5324.2 1973.69  5366.7 1982.08  5438.2 1990.92  5565.6 1995.74
  5741.8 2003.35  5855.3 2011.67  5945.9 2014.92  6219.4 2018.24  6490.3 2015.31
#Mann= 16 ,-1 , 0
  4030.6      .1       0  4180.9     .16       0  4254.3     .05       0
  4317.4     .16       0  4384.6     .05       0  4467.6     .16       0
    4654     .05       0  4680.5     .16       0  4826.5      .1       0
  4974.6     .07       0  4980.6      .1       0    5296     .16       0
  5438.2      .1       0  5565.6     .16       0  5741.8      .1       0
  6219.4     .16       0
Bank Sta=4906.8,5055.2
XS Rating Curve= 0 ,0
Exp/Cntr=0.3,0.1

Type RM Length L Ch R = 1 ,52147   ,339,339,339
BEGIN DESCRIPTION:
WHITE OAK CREEK 78.0
END DESCRIPTION:
XS GIS Cut Line= 3
      2672976.99     10033820.36      2673862.43     10033153.68
      2674065.56     10032351.57
#Sta/Elev= 30
    4110 1995.24  4244.5 1983.79  4300.7 1976.84  4394.4 1972.79  4515.2 1956.84
  4594.3 1942.14  4629.7 1940.11  4663.4 1939.09  4779.6 1938.12  4844.2 1933.97
  4950.5 1932.48  4979.5  1928.9  4997.6 1921.98  5000.4 1921.48  5003.6 1921.98
  5037.8 1928.63  5064.9 1926.09  5108.6 1925.61  5129.4 1927.97 5147.73 1932.52
  5158.6  1937.8  5463.9  1942.3  5496.8 1944.69  5527.4 1950.75  5558.7 1960.37
  5627.9 1975.21  5727.5 1979.16  5750.9 1982.07  5832.8 1986.49  6045.8  1993.7
#Mann= 7 ,-1 , 0
    4110      .1       0  4629.7     .16       0  4663.4      .1       0
  4997.6     .07       0  5003.6      .1       0  5527.4     .16       0
  5727.5      .1       0
Bank Sta=4950.5,5147.73
XS Rating Curve= 0 ,0
Exp/Cntr=0.3,0.1

Type RM Length L Ch R = 1 ,51808   ,429,429,429
BEGIN DESCRIPTION:
WHITE OAK CREEK 77.0
END DESCRIPTION:
XS GIS Cut Line= 3
      2673154.14     10033940.12      2673773.89     10033617.22
       2674903.8     10032909.07
#Sta/Elev= 30
  4174.8 1996.85  4302.9 1987.65  4356.2 1981.12  4435.4  1973.6  4574.3 1939.19
  4631.1 1935.81  4783.4 1934.45  4805.5 1930.93  4811.1 1929.32  4871.7 1926.49
  4966.2 1927.89  4999.8 1920.31  5002.5 1919.81  5005.8 1920.31    5024 1921.67
  5039.3 1930.64  5060.5 1936.05  5162.3 1932.34  5227.9 1936.49  5395.2 1937.55
  5445.5 1944.89  5510.7 1945.53  5547.2 1952.06  5605.9 1957.08  5678.1 1963.33
    5757 1974.29  5823.2 1979.26  5872.5 1985.62  6134.2 2005.35  6207.1 2014.01
#Mann= 6 ,-1 , 0
  4174.8      .1       0  4356.2     .16       0  4631.1      .1       0
  4999.8     .07       0  5005.8      .1       0  5605.9     .16       0
Bank Sta=4805.5,5039.3
XS Rating Curve= 0 ,0
Exp/Cntr=0.3,0.1

Type RM Length L Ch R = 1 ,51379   ,385,385,385
BEGIN DESCRIPTION:
WHITE OAK CREEK 76.0
END DESCRIPTION:
XS GIS Cut Line= 3
      2673263.51      10034106.8      2674461.39      10033851.6
      2675070.76     10033565.14
#Sta/Elev= 30
  4247.9 2003.72  4282.6 2002.69  4332.1 1996.85  4396.1 1994.87  4437.9 1991.42
  4518.8 1985.59  4569.7 1978.91  4610.8 1968.05  4682.4 1941.44  4702.8 1935.65
  4718.4 1933.11  4774.4 1931.12  4834.7 1932.05  4861.9 1933.06  4876.7 1931.47
  4897.1 1926.79    4938 1920.81  4968.7 1922.19  4996.4 1918.56  4999.1 1918.06
  5002.4 1918.56  5019.8 1920.33  5040.2 1927.42  5099.5 1927.71  5132.3 1930.07
  5613.1  1936.6  5845.1 1946.76  5921.5 1955.21  6063.8 1974.66    6146 1983.39
#Mann= 5 ,-1 , 0
  4247.9      .1       0  4437.9     .16       0  4834.7      .1       0
  4996.4     .07       0  5002.4      .1       0
Bank Sta=4897.1,5040.2
XS Rating Curve= 0 ,0
Exp/Cntr=0.3,0.1

Type RM Length L Ch R = 1 ,50994   ,280,280,280
BEGIN DESCRIPTION:
WHITE OAK CREEK 75.0
END DESCRIPTION:
XS GIS Cut Line= 4
      2673409.31     10034429.72      2674060.35      10034356.8
      2674398.89     10034096.39      2675221.84     10033872.42
#Sta/Elev= 30
  4235.7 1993.68  4365.7 1982.37  4467.2 1963.83  4496.5  1957.5  4512.8 1951.48
  4517.9 1951.99  4566.9 1937.92    4603  1932.3  4648.8 1930.34  4768.2 1928.54
  4873.7 1929.69  4882.1 1927.03  4899.4  1919.7  4905.7 1919.11  4934.7 1919.93
    4970 1917.44  5002.4 1917.36  5005.1 1916.86  5008.4 1917.36  5034.4 1922.28
  5090.5 1924.68    5105 1927.02  5127.7 1932.03  5163.1 1933.35  5524.8 1932.98
  5721.7 1937.47  5835.7 1942.82    5921 1952.45  6123.3 1993.03  6170.8 2000.41
#Mann= 6 ,-1 , 0
  4235.7      .1       0  4467.2     .16       0  4648.8      .1       0
  5002.4     .07       0  5008.4      .1       0  6123.3     .16       0
Bank Sta=4882.1,5105
XS Rating Curve= 0 ,0
Exp/Cntr=0.3,0.1

Type RM Length L Ch R = 1 ,50714   ,610,610,610
BEGIN DESCRIPTION:
WHITE OAK CREEK 74.0
END DESCRIPTION:
XS GIS Cut Line= 3
      2673409.27     10034492.22      2674393.68     10034575.55
      2675232.22      10034169.3
#Sta/Elev= 30
  4221.3 1989.37  4290.7 1984.89  4411.2 1968.79  4481.2  1955.6  4541.6 1939.45
  4581.8 1934.31  4635.6 1931.98  4770.1 1927.23  4894.6 1926.29    4933 1925.39
  4963.1 1918.72  5000.3 1915.87    5003 1915.37  5006.3 1915.87  5053.5    1921
 5068.18 1926.16  5083.6  1930.8  5103.6 1932.53    5194 1928.46  5312.8 1930.75
  5325.7 1928.81  5386.1 1929.68  5403.1  1928.4  5836.8 1934.65  5916.5 1941.87
    5989 1962.09  6023.9 1972.46  6074.6 1982.68  6091.6 1988.13    6141 1997.21
#Mann= 6 ,-1 , 0
  4221.3      .1       0  4481.2     .16       0  4635.6      .1       0
  5000.3     .07       0  5006.3      .1       0    5989     .16       0
Bank Sta=4894.6,5068.18
XS Rating Curve= 0 ,0
Exp/Cntr=0.3,0.1

Type RM Length L Ch R = 1 ,50104   ,622,622,622
BEGIN DESCRIPTION:
WHITE OAK CREEK 73.0
END DESCRIPTION:
XS GIS Cut Line= 3
      2673044.67     10034966.17      2674247.85      10035164.1
      2675331.17     10034471.39
#Sta/Elev= 30
    4013 2006.91  4130.4 2001.63    4331 1993.06  4442.5 1984.05    4635  1956.9
  4746.5 1932.38  4939.1 1924.28  4953.6 1923.22  4979.6 1913.37  4996.9 1912.98
  4999.6 1912.48  5002.9 1912.98  5070.8 1918.01  5091.1 1922.19  5137.2 1923.82
  5637.4 1929.73  5921.5 1926.35  6079.7 1931.72  6116.1 1935.69  6130.9 1940.06
  6152.4 1942.31  6188.8 1955.71  6246.3 1966.69  6261.5 1973.12  6282.7 1974.99
  6297.9 1980.03    6319 1980.92  6334.3 1986.46  6391.8 1996.09  6518.2 2004.45
#Mann= 5 ,-1 , 0
    4013     .16       0  4130.4      .1       0  4996.9     .07       0
  5002.9      .1       0  6130.9     .16       0
Bank Sta=4939.1,5137.2
XS Rating Curve= 0 ,0
Exp/Cntr=0.3,0.1

Type RM Length L Ch R = 1 ,49482   ,375,375,375
BEGIN DESCRIPTION:
WHITE OAK CREEK 72.0
END DESCRIPTION:
XS GIS Cut Line= 4
      2673835.52     10036490.48      2674259.13     10035823.82
      2674307.74     10035309.93      2675300.84     10034712.68
#Sta/Elev= 30
    3951 1964.99  4247.4 1946.21  4262.6 1943.07  4283.8  1942.2  4314.3 1936.14
  4341.4 1936.26  4371.9 1932.23  4690.3 1924.69  4851.4 1924.32  4911.7 1921.04
    4972 1911.34  5019.2 1910.49  5021.9 1909.99  5025.2 1910.49  5092.5 1919.53
  5182.9 1921.26    5415 1925.01  5946.4 1925.54  6028.1 1930.19  6056.1 1934.56
  6090.4 1945.13  6114.3 1950.93  6129.9 1958.22  6151.2 1964.95  6172.6 1968.73
  6188.2 1974.22  6230.9 1980.38  6246.4 1984.82  6326.1 1992.98  6415.9 1996.52
#Mann= 4 ,-1 , 0
    3951      .1       0  5019.2     .07       0  5025.2      .1       0
  6090.4     .16       0
Bank Sta=4911.7,5182.9
XS Rating Curve= 0 ,0
Exp/Cntr=0.3,0.1

Type RM Length L Ch R = 1 ,49107   ,461,461,461
BEGIN DESCRIPTION:
WHITE OAK CREEK 71.0
END DESCRIPTION:
XS GIS Cut Line= 4
      2673932.73     10036636.33      2674599.41     10035948.82
      2674661.91     10035427.99      2675411.89     10034823.83
#Sta/Elev= 30
  3735.7 1962.99  3953.7 1949.05  4073.9 1944.87  4335.7 1930.91  4497.2 1926.87
  4522.8 1926.62  4682.4 1922.39  4738.8 1919.86  4798.6 1917.67  4977.4 1910.52
  4982.4 1911.79  4997.7 1908.48  5000.4 1907.98  5003.7 1908.48  5020.8  1909.7
  5064.6 1918.52  5131.6 1919.77  5232.7 1922.76  5389.5 1922.49  5439.1 1924.25
  5659.8 1925.12  5701.5 1928.91  5752.1  1944.6  5773.4 1952.34    5823  1966.5
  5837.4 1972.63  5901.4 1983.83  5965.3 1988.66  6107.7 1995.85    6181 1996.58
#Mann= 8 ,-1 , 0
  3735.7      .1       0  4497.2     .16       0  4522.8      .1       0
  4682.4     .16       0  4798.6      .1       0  4997.7     .07       0
  5003.7      .1       0  5752.1     .16       0
Bank Sta=4738.8,5131.6
XS Rating Curve= 0 ,0
Exp/Cntr=0.3,0.1

Type RM Length L Ch R = 1 ,48646   ,778,778,778
BEGIN DESCRIPTION:
WHITE OAK CREEK 70.0
END DESCRIPTION:
XS GIS Cut Line= 2
      2673884.15      10036886.3      2675418.83     10035539.11
#Sta/Elev= 30
  3526.5 1972.55  3538.4 1973.38  3552.7 1970.33  3581.1 1967.61  3587.8 1968.43
  3616.3 1963.64  3677.7 1961.46  3722.5 1960.05  3793.7 1953.83  4119.2 1940.17
  4155.2 1940.02  4417.1 1924.59  4664.8 1921.01    4736 1917.77  4913.4 1913.81
  4962.8 1908.32  4994.9 1907.75  4997.6 1907.25  5000.9 1907.75  5012.1 1909.45
  5033.9 1918.05  5054.8 1920.19  5224.7 1915.57  5247.6 1919.07  5281.6 1931.91
  5295.8 1942.02  5324.3 1954.29  5402.1 1973.69  5479.9 1974.55  5568.6 1971.84
#Mann= 5 ,-1 , 0
  3526.5     .05       0  3677.7      .1       0  4994.9     .07       0
  5000.9      .1       0  5247.6     .16       0
#XS Ineff= 1 ,-1
  5055.4 5342.33 1920.33
Permanent Ineff=
       F
Bank Sta=4736,5033.9
XS Rating Curve= 0 ,0
Exp/Cntr=0.3,0.1

Type RM Length L Ch R = 1 ,47868   ,979,979,979
BEGIN DESCRIPTION:
WHITE OAK CREEK 68.0
END DESCRIPTION:
XS GIS Cut Line= 4
      2674550.79      10037830.8      2674745.24     10036921.04
      2675509.13      10036476.6      2675856.34     10035573.85
#Sta/Elev= 30
  3480.8 1978.95    3621 1972.95  3780.1 1959.82  4020.9 1949.02  4160.6 1941.53
  4210.1 1936.02  4290.9 1922.46  4326.6 1918.21  4354.2 1919.39  4377.7 1920.94
  4402.9 1917.34  4551.4 1915.29  4754.9 1915.52  4872.4 1911.88  4899.8 1911.56
  4974.2 1909.94  4989.9 1904.08  5001.9 1902.84  5004.6 1902.34  5007.9 1902.84
  5091.7 1912.14  5114.5 1914.64  5134.7 1917.37  5297.9 1921.05  5613.6  1934.4
    5783 1939.85  5929.7 1950.86  6170.8 1973.55    6214 1974.91  6262.1 1976.91
#Mann= 12 ,-1 , 0
  3480.8     .16       0  4020.9      .1       0  4290.9     .05       0
  4354.2      .1       0  4899.8     .05       0  5001.9    .035       0
  5007.9     .05       0  5114.5      .1       0  5297.9     .05       0
  5613.6      .1       0  5929.7     .16       0    6214      .1       0
Bank Sta=4872.4,5091.7
XS Rating Curve= 0 ,0
Exp/Cntr=0.3,0.1

Type RM Length L Ch R = 1 ,46889   ,713,713,713
BEGIN DESCRIPTION:
WHITE OAK CREEK 67.0
END DESCRIPTION:
XS GIS Cut Line= 3
      2675446.63     10038296.01      2675585.52     10036761.32
      2675932.58     10035588.24
#Sta/Elev= 30
  4219.4 2008.94  4442.6 2002.67  4517.5 1998.64  4628.2 1989.77  4763.9 1974.45
  4849.6 1961.57  4894.4 1958.75  4904.5 1951.68  4914.5 1930.48  4924.5 1920.42
  4944.6 1913.15  4954.7 1909.03  4960.3 1904.01  4994.6 1898.01    5035  1900.3
  5055.1 1907.56    5071 1908.78  5168.5 1911.45  5266.9 1910.57  5309.8 1911.23
    5501 1911.99  6000.2 1919.15  6026.3 1920.09  6179.3  1925.5  6275.3 1929.97
  6361.6 1933.31    6569 1946.32  6852.8 1974.14  6919.4 1976.84  6983.7 1981.61
#Mann= 13 ,-1 , 0
  4219.4     .16       0  4944.6     .07       0  5168.5      .1       0
  5266.9     .05       0  5309.8      .1       0    5501     .05       0
  6000.2      .1       0  6026.3     .05       0  6179.3      .1       0
  6275.3     .05       0  6361.6      .1       0    6569     .16       0
  6919.4      .1       0
Bank Sta=4954.7,5071
XS Rating Curve= 0 ,0
Exp/Cntr=0.3,0.1

Type RM Length L Ch R = 1 ,46176   ,1031,1031,1031
BEGIN DESCRIPTION:
WHITE OAK CREEK 65.0
END DESCRIPTION:
XS GIS Cut Line= 3
      2675835.51     10038455.78      2676217.46     10037629.37
      2676120.24     10035483.58
#Sta/Elev= 30
    3884    1997  3957.4 1996.99  4000.7 1996.41  4213.1 1990.58  4355.1 1986.07
  4518.7 1974.22  4602.3 1961.62  4630.3 1959.48  4794.4 1940.22  4831.7 1934.02
  4840.1 1934.32  4870.1 1927.42  4920.2    1906    5000 1896.13  5020.3 1897.98
  5050.3 1905.27  5090.3 1908.09  5110.4 1906.68  5210.5 1905.78  5363.7 1909.88
  5457.9  1909.7    5721 1908.65  5931.8 1911.45  6030.5  1914.5  6177.4 1923.17
  6326.5 1933.39  6622.5    1969  6782.1 1987.72  6869.2  1995.1  6942.4 1997.69
#Mann= 15 ,-1 , 0
    3884     .16       0  3957.4      .1       0  4000.7     .16       0
  4213.1      .1       0  4518.7     .05       0  4630.3      .1       0
  4831.7     .07       0  5110.4     .05       0  5363.7      .1       0
  5457.9     .05       0  5931.8      .1       0  6030.5     .05       0
  6177.4      .1       0  6326.5     .16       0  6622.5      .1       0
Bank Sta=4920.2,5090.3
XS Rating Curve= 0 ,0
Exp/Cntr=0.3,0.1

Type RM Length L Ch R = 1 ,45145   ,490,490,490
BEGIN DESCRIPTION:
WHITE OAK CREEK 63.0
END DESCRIPTION:
XS GIS Cut Line= 4
      2677085.52     10038171.06      2677252.19     10037108.54
      2676786.91     10036566.87      2676509.12     10035712.69
#Sta/Elev= 30
  3524.5 1979.26  3744.5 1972.93  3786.5 1969.38  3898.8 1960.07  3946.9 1956.37
  4025.2 1945.87    4200 1930.27  4830.7 1903.71  4946.8 1904.77    4961 1903.06
  4973.7 1896.46  4993.2 1893.48  4995.9 1892.98  4999.2 1893.48  5024.7 1895.73
    5039 1899.92  5100.9 1900.53  5108.5 1901.28  5159.7 1903.46  5197.6 1904.34
  5783.6 1905.77  5840.2 1910.26  5864.2 1918.02  5904.1 1934.94  5936.1 1943.44
  6005.2 1952.45  6031.9 1958.67  6069.1  1961.9    6133 1972.68  6212.3 1982.64
#Mann= 11 ,-1 , 0
  3524.5      .1       0  3786.5     .16       0  3898.8      .1       0
  4830.7     .05       0  4973.7      .1       0  4993.2     .07       0
  4999.2      .1       0  5100.9     .05       0  5108.5      .1       0
  5197.6     .05       0  5783.6     .16       0
Bank Sta=4961,5159.7
XS Rating Curve= 0 ,0
Exp/Cntr=0.3,0.1

Type RM Length L Ch R = 1 ,44655   ,615,615,615
BEGIN DESCRIPTION:
WHITE OAK CREEK 62.0
END DESCRIPTION:
XS GIS Cut Line= 3
      2677867.63     10037965.29      2677687.08      10037041.7
      2676694.04     10035611.16
#Sta/Elev= 30
  3284.5 1965.65  3406.8 1953.61  3520.4 1940.28  3805.7 1924.58  4379.7  1910.6
  4442.2 1909.29  4527.4  1907.8  4583.9 1906.82  4690.2 1902.38  4704.7    1901
  4791.8 1900.08  4847.9 1900.32  4955.2 1894.01  4984.9 1896.79  5002.9 1891.98
  5005.6 1891.48  5008.9 1891.98  5027.4 1899.82  5035.6 1901.81  5184.6 1900.16
  5197.3    1900  5503.8 1901.88  5571.8 1904.59  5596.2 1906.59  5623.2 1914.11
  5652.9  1924.3  5709.6 1950.56  5739.4 1959.85  5825.8  1978.5    5967 1996.48
#Mann= 15 ,-1 , 0
  3284.5     .16       0  3406.8      .1       0  4379.7     .05       0
  4442.2      .1       0  4527.4     .05       0  4583.9      .1       0
  4690.2     .16       0  4791.8      .1       0  5002.9     .07       0
  5008.9      .1       0  5027.4     .05       0  5184.6      .1       0
  5197.3     .05       0  5503.8      .1       0  5571.8     .16       0
Bank Sta=4704.7,5035.6
XS Rating Curve= 0 ,0
Exp/Cntr=0.3,0.1
