HEC-RAS study WHITE OAK CREEK.prj: WHITE OAK CREEK Base Level Engineering

--- WHITE OAK CREEK.g01 (geometry) --- (continued)

Type RM Length L Ch R = 1 ,44040   ,2042,2042,2042
BEGIN DESCRIPTION:
WHITE OAK CREEK 61.0
END DESCRIPTION:
XS GIS Cut Line= 3
      2678478.75     10037173.64      2677624.58     10035909.76
      2676666.23     10035222.25
#Sta/Elev= 30
  3729.4 1942.95    3809 1931.04  3952.9 1916.21    4161 1906.71  4324.5 1903.46
  4495.2 1902.69  4757.6  1901.3    4888 1899.74  4917.8 1895.83  4974.8    1895
  4993.6 1889.05  4996.3 1888.55  4999.6 1889.05  5040.7 1896.81  5061.7 1897.83
  5184.2 1896.36  5570.8 1897.02  5650.6 1899.54  5690.1 1900.69  5691.9 1900.77
  5736.6 1902.81  5786.9 1910.42  5816.2 1920.97    5879 1955.86  5929.4 1979.82
  5958.9 1987.95  6002.7 1994.97  6095.2 1998.04  6373.9 1999.82  6434.3  2002.9
#Mann= 11 ,-1 , 0
  3729.4      .1       0    4161     .05       0  4324.5      .1       0
  4495.2     .05       0  4757.6      .1       0  4993.6     .07       0
  4999.6      .1       0  5184.2     .16       0  5690.1      .1       0
  5691.9     .16       0  6002.7      .1       0
Bank Sta=4888,5650.6
XS Rating Curve= 0 ,0
Exp/Cntr=0.3,0.1

Type RM Length L Ch R = 1 ,41998   ,395,395,395
BEGIN DESCRIPTION:
WHITE OAK CREEK 58.0
END DESCRIPTION:
XS GIS Cut Line= 3
      2678575.97     10037243.07      2678735.69     10035263.92
      2678235.69     10033923.63
#Sta/Elev= 30
  3211.1 1958.43  3394.5 1933.37  3465.5 1927.12  3591.7 1916.75  3677.1 1913.07
    4013 1901.96  4143.5  1900.6  4193.6 1896.17    4393 1892.93  4421.2 1892.34
  4582.8 1891.18    4676 1888.75  4745.4 1891.18    4926 1890.61  4966.1  1889.2
  4976.2 1885.41    5006 1882.17  5016.3 1886.62  5076.5 1892.26  5106.6 1895.92
  5282.3 1905.11  5404.2 1915.57  5429.1 1923.67  5581.1 1942.06  5783.9 1958.77
    6089 1969.51  6149.7 1974.02  6401.1 1975.58    6605 1980.57  6627.2 1982.13
#Mann= 8 ,-1 , 0
  3211.1      .1       0  3394.5     .05       0  3465.5      .1       0
    4393     .05       0  4582.8      .1       0  4745.4     .07       0
  5076.5      .1       0    6605     .16       0
Bank Sta=4421.2,5076.5
XS Rating Curve= 0 ,0
Exp/Cntr=0.3,0.1

Type RM Length L Ch R = 1 ,41603   ,780,780,780
BEGIN DESCRIPTION:
WHITE OAK CREEK 57.0
END DESCRIPTION:
XS GIS Cut Line= 3
      2678791.26     10037097.21       2679159.3     10035250.03
      2679076.11     10034307.18
#Sta/Elev= 30
  3435.2 1944.83  3457.8 1942.61  3547.3 1931.69  3702.7 1921.27    3956 1907.76
  4471.9 1897.43  4580.8 1890.59  4595.6 1889.55  4747.7 1888.06  4803.6 1888.35
  4845.9 1889.45  4927.9 1887.22  4981.8 1885.52  4995.8 1879.74  4998.6 1879.24
  5001.8 1879.74  5023.8 1884.81    5060 1890.93  5289.1 1892.03  5553.8 1901.66
  5616.9 1903.75    5729 1915.55  5816.9  1935.6  5907.3 1947.57  5953.2  1956.5
  5972.1 1957.72  6065.3 1970.41  6070.3  1968.9    6108  1973.8  6265.2  1979.3
#Mann= 12 ,-1 , 0
  3435.2      .1       0  3457.8     .05       0  3702.7      .1       0
  4595.6     .05       0  4747.7      .1       0  4803.6     .05       0
  4927.9      .1       0  4995.8     .07       0  5001.8      .1       0
  5023.8     .05       0  5553.8      .1       0  5972.1     .16       0
Bank Sta=4580.8,5060
XS Rating Curve= 0 ,0
Exp/Cntr=0.3,0.1

Type RM Length L Ch R = 1 ,40823   ,1692,1692,1692
BEGIN DESCRIPTION:
WHITE OAK CREEK 56.0
END DESCRIPTION:
XS GIS Cut Line= 4
      2679360.67     10037298.69      2679832.91     10036347.26
       2679534.3     10035534.76      2679173.32     10034222.73
#Sta/Elev= 30
    3559 1951.98    4100 1922.02  4705.7 1901.27  4891.3 1897.69    4964 1891.61
  4969.3 1894.14 4983.52 1888.39  4987.2 1886.76  4991.5 1878.31  4994.2 1877.81
  5072.4 1882.99  5141.5 1882.11  5258.1 1887.85  5264.2 1887.97    5519  1885.1
  5679.1 1887.11  5894.5 1889.81  5988.6 1891.63  6042.8 1893.13  6088.7 1894.63
  6133.5 1902.72  6202.3 1909.55  6283.8 1928.97  6400.6 1954.83    6495 1970.05
  6535.4 1976.62    6571 1977.88  6696.2 1986.57  6774.4 1987.34  6847.6 1988.56
#Mann= 11 ,-1 , 0
    3559      .1       0 4983.52     .07       0  5258.1      .1       0
  5679.1     .05       0  5894.5      .1       0  5988.6     .05       0
  6042.8      .1       0  6283.8     .16       0    6495      .1       0
    6571     .16       0  6774.4      .1       0
Bank Sta=4983.52,5264.2
XS Rating Curve= 0 ,0
Exp/Cntr=0.3,0.1

Type RM Length L Ch R = 1 ,39131   ,1043,1043,1043
BEGIN DESCRIPTION:
WHITE OAK CREEK 55.0
END DESCRIPTION:
XS GIS Cut Line= 3
      2679935.78     10036487.45      2680289.95     10034876.34
      2679735.01      10034057.8
#Sta/Elev= 30
  2955.8 1910.19  3315.2 1899.09  3773.8  1892.4    4080 1889.62  4126.8  1890.3
  4279.5  1885.5  4430.4  1885.8  4644.8 1885.92  4738.5 1884.63  4795.5 1881.38
  4852.4 1878.35  4945.7 1877.15  4969.1 1877.25  4987.1 1874.38  4989.9 1873.88
  4993.1 1874.38  5032.1 1874.79    5041 1876.78  5051.2 1881.71  5068.1  1886.6
  5148.8  1886.3  5220.7 1890.55  5235.7 1893.13  5271.6 1901.59  5292.6 1909.02
  5385.5 1951.63  5406.5 1960.33  5457.4 1977.33  5529.3 1985.94  5594.3 1986.86
#Mann= 9 ,-1 , 0
  2955.8      .1       0  3773.8     .05       0    4080      .1       0
  4279.5     .05       0  4430.4      .1       0  4945.7     .16       0
  4987.1     .07       0  4993.1     .16       0  5051.2      .1       0
Bank Sta=4795.5,5051.2
XS Rating Curve= 0 ,0
Exp/Cntr=0.3,0.1

Type RM Length L Ch R = 1 ,38088   ,847,847,847
BEGIN DESCRIPTION:
WHITE OAK CREEK 54.0
END DESCRIPTION:
XS GIS Cut Line= 4
      2680032.99     10036431.92      2680810.78     10034279.11
      2681324.67     10034084.67      2681199.73      10031967.7
#Sta/Elev= 30
  2581.8 1909.24  2718.1 1907.37  3022.9 1896.99  3493.6 1893.64  3688.7 1892.47
  3738.8 1892.86  3782.5  1889.8  3997.6  1883.3  4262.9 1883.47  4528.3 1880.77
  4586.1 1878.24  4738.3 1876.81  4918.8 1867.84  4921.5 1867.34  4924.8 1867.84
  4957.9 1871.21  5012.9 1870.22  5037.7 1873.79  5043.1 1876.45  5060.8 1879.43
  5133.2 1878.33  5329.2    1879  5778.5 1876.65  6272.2 1880.39    6453 1883.18
  6583.2 1894.99  6822.3 1903.38  7130.6 1918.67  7425.4 1930.51  7540.9 1934.26
#Mann= 13 ,-1 , 0
  2581.8      .1       0  3493.6     .05       0  3688.7      .1       0
  3782.5     .05       0  4586.1      .1       0  4918.8     .07       0
  4924.8      .1       0  5133.2     .16       0  5329.2      .1       0
  6272.2     .16       0  6822.3      .1       0  7130.6     .05       0
  7425.4      .1       0
#XS Ineff= 1 ,-1
 5068.98 6456.78 1879.82
Permanent Ineff=
       F
Bank Sta=4738.3,5043.1
XS Rating Curve= 0 ,0
Exp/Cntr=0.3,0.1

Type RM Length L Ch R = 1 ,37681   ,438,438,438
BEGIN DESCRIPTION:
Mapping XS e712f7ec
END DESCRIPTION:
XS GIS Cut Line= 4
      2680129.01     10036424.76      2681129.03     10034586.18
      2681483.19     10034164.31      2681394.67      10032128.3
#Sta/Elev= 30
  2812.3 1908.46  2958.1 1907.46  3005.1  1904.8  3280.6 1897.27    3512 1895.67
  3645.6 1894.85  4016.3 1893.11  4058.2 1892.86  4184.6 1884.93    4649 1880.83
  4723.2 1880.57  4832.4 1872.62  4870.4 1874.58  4948.7 1871.72  4977.3 1864.71
  5002.9 1864.21  5005.7 1863.71  5008.9 1864.21  5026.7 1867.32  5041.1 1873.73
  5055.4 1878.73  5069.7 1879.56  5967.1 1874.26  6397.5 1879.55  6457.6 1881.51
  6497.6 1888.05  6547.7 1892.36    6827 1896.36  7248.3 1919.34    7494 1924.78
#Mann= 11 ,-1 , 0
  2812.3      .1       0  2958.1     .05       0  3005.1      .1       0
  3280.6     .05       0    3512      .1       0  3645.6     .05       0
  4016.3      .1       0  4184.6     .05       0    4649      .1       0
  5002.9     .07       0  5008.9      .1       0
Bank Sta=4948.7,5041.1
XS Rating Curve= 0 ,0
Exp/Cntr=0.3,0.1

Type RM Length L Ch R = 1 ,37243   ,1015,1015,1015
BEGIN DESCRIPTION:
WHITE OAK CREEK 53.0
END DESCRIPTION:
XS GIS Cut Line= 4
      2680174.12     10036405.88      2681363.33     10035129.87
      2681979.65     10033584.73      2682864.26     10032951.62
#Sta/Elev= 30
  2892.6 1907.46  2992.1 1906.77  3135.9 1903.37  3334.5 1899.02  3551.5 1896.09
  3578.3 1895.81  4931.9 1887.52  4955.7 1881.66  4961.1 1871.24  4977.2 1862.75
  4987.7 1862.39  4990.5 1861.89  4993.7 1862.39  5074.3 1864.09  5176.7 1873.55
  5386.3 1875.07  5461.7 1866.22  5721.2 1874.95  6075.4 1874.39  6107.7 1866.54
    6183 1873.11  6342.3 1873.32    6502 1873.52  6622.4 1879.56  6687.5 1894.78
  6758.7  1898.2  6938.4 1944.61  7052.4 1966.79  7138.4 1977.86  7388.2 1978.06
#Mann= 11 ,-1 , 0
  2892.6      .1       0  2992.1     .05       0  3135.9      .1       0
  3334.5     .05       0  3551.5      .1       0  3578.3     .05       0
  4931.9      .1       0  4987.7     .07       0  4993.7      .1       0
  6342.3     .16       0    6502      .1       0
#XS Ineff= 2 ,-1
 5312.68 5762.25 1876.52    6080 6708.73 1874.72
Permanent Ineff=
       F       F
Bank Sta=4955.7,5176.7
XS Rating Curve= 0 ,0
Exp/Cntr=0.3,0.1

Type RM Length L Ch R = 1 ,36228   ,979,979,979
BEGIN DESCRIPTION:
WHITE OAK CREEK 52.0
END DESCRIPTION:
XS GIS Cut Line= 5
      2680248.27     10036424.95       2682345.5     10034737.45
      2682359.39     10034056.89       2683220.5     10033348.56
      2684053.68     10033369.39
#Sta/Elev= 30
  1975.1 1907.53  2042.6 1906.83  2368.7 1900.76  2447.9 1899.48  2613.2 1896.77
  2758.7 1894.63  3012.3 1891.56  3026.3 1891.43  3725.6 1887.76  4244.2 1878.47
  4515.8 1871.09  4940.7 1864.33  4997.7 1855.47  5000.5 1854.97  5003.7 1855.47
  5030.7 1869.21  5540.7 1868.95  5626.5 1862.73  5655.2 1875.11  5768.5 1893.46
  5939.3 1891.86  5974.4 1895.39  5988.8  1902.9  6023.9  1904.7  6052.6 1913.42
  6229.8 1932.12  6272.9  1943.7  6500.6 1976.41  6660.7 1988.76  7296.1 2014.76
#Mann= 11 ,-1 , 0
  1975.1      .1       0  2042.6     .05       0  2368.7      .1       0
  2447.9     .05       0  2613.2      .1       0  2758.7     .05       0
  3012.3      .1       0  3026.3     .05       0  4244.2      .1       0
  4997.7     .07       0  5003.7      .1       0
#XS Ineff= 1 ,-1
 5040.57 5763.06 1870.29
Permanent Ineff=
       F
Bank Sta=4515.8,5030.7
XS Rating Curve= 0 ,0
Exp/Cntr=0.3,0.1

Type RM Length L Ch R = 1 ,35249   ,943,943,943
BEGIN DESCRIPTION:
WHITE OAK CREEK 50.0
END DESCRIPTION:
XS GIS Cut Line= 2
      2680442.72     10036438.84      2683880.22     10034570.78
#Sta/Elev= 30
  2029.6 1906.52  2886.3 1891.54  3186.5 1890.15  3704.4 1882.06  4020.8 1882.98
  4073.4  1881.1  4080.7 1877.76  4102.5 1875.19  4140.5 1873.19  4544.4 1872.18
  4685.9 1865.83  4729.6 1862.85  4942.5 1863.44  4972.5  1861.2  4995.3  1854.5
  5007.8 1853.73  5040.4 1856.94  5074.9 1868.46  5084.1 1873.75  5127.8 1906.43
  5143.2 1915.33  5177.4 1956.32  5200.1 1968.78  5222.9  1979.2  5253.2 1988.49
  5332.2 1990.71  5541.6 1988.19    5695 1978.52  5864.2 1980.34  5941.9 1985.69
#Mann= 4 ,-1 , 0
  2029.6      .1       0  4685.9     .07       0  5084.1     .16       0
  5332.2      .1       0
Bank Sta=4942.5,5074.9
XS Rating Curve= 0 ,0
Exp/Cntr=0.3,0.1

Type RM Length L Ch R = 1 ,34306   ,1078,1078,1078
BEGIN DESCRIPTION:
WHITE OAK CREEK 48.0
END DESCRIPTION:
XS GIS Cut Line= 4
      2680664.97      10036466.6      2682824.67     10035681.89
      2683296.89     10036001.34      2683491.35     10035945.78
#Sta/Elev= 30
  2347.2 1903.93  2477.2 1902.72  2498.6 1902.74  2657.5 1900.08  2832.4 1895.43
  2875.6 1894.98    3050 1890.96  3101.8 1890.37  3246.2 1888.16  3799.9 1882.93
  3989.4 1878.63  4155.4 1870.67  4537.3 1862.75  4593.1 1860.38  4839.1 1859.15
  4902.1 1858.69  4933.2 1852.64  4998.1 1851.28  5000.8 1850.78  5004.1 1851.28
    5041 1858.35  5060.1 1864.23  5123.9  1878.4  5159.9 1893.83  5174.8 1904.81
  5216.9 1925.77  5257.1 1945.16  5274.2 1949.04  5341.6 1960.12  5417.4 1956.66
#Mann= 18 ,-1 , 0
  2347.2     .05       0  2477.2      .1       0  2498.6     .05       0
  2657.5      .1       0  2832.4     .05       0  2875.6      .1       0
    3050     .05       0  3101.8      .1       0  3246.2     .05       0
  3799.9      .1       0  4593.1     .16       0  4839.1      .1       0
  4933.2     .16       0  4998.1     .07       0  5004.1     .16       0
    5041      .1       0  5216.9     .16       0  5274.2      .1       0
Bank Sta=4537.3,5060.1
XS Rating Curve= 0 ,0
Exp/Cntr=0.3,0.1

Type RM Length L Ch R = 1 ,33228   ,754,754,754
BEGIN DESCRIPTION:
WHITE OAK CREEK 47.0
END DESCRIPTION:
XS GIS Cut Line= 4
      2680685.78     10036924.95      2681880.22     10036626.34
       2682845.5     10036751.34      2683428.84     10036195.78
#Sta/Elev= 30
  3185.1 1908.84  3237.9  1907.9  3516.1  1900.3  3862.6 1891.15  4257.4 1885.35
  4361.5 1881.58  4432.3 1871.03  4535.5 1863.98  4662.1 1859.87  4849.5 1858.73
    4949 1860.24    4959 1857.45  4969.1 1850.23  4986.3  1847.6    4989  1847.1
  4992.3  1847.6  5056.4 1853.82  5110.3 1854.96  5140.7 1852.17  5289.8  1856.5
  5479.6 1857.18  5530.5 1857.82  5559.6 1858.33  5672.9 1861.58  5772.9 1868.96
  5934.6 1900.27    6030 1922.85  6097.5 1943.66  6159.8 1958.18  6195.2 1960.62
#Mann= 15 ,-1 , 0
  3185.1      .1       0  3237.9     .05       0  3516.1      .1       0
  3862.6     .05       0  4257.4      .1       0  4662.1     .05       0
  4849.5      .1       0  4986.3     .07       0  4992.3      .1       0
  5289.8     .16       0  5479.6      .1       0  5530.5     .05       0
  5772.9      .1       0    6030     .16       0  6159.8      .1       0
#XS Ineff= 1 ,-1
 4477.56 4948.86  1860.5
Permanent Ineff=
       F
Bank Sta=4959,5559.6
XS Rating Curve= 0 ,0
Exp/Cntr=0.3,0.1

Type RM Length L Ch R = 1 ,32474   ,497,497,497
BEGIN DESCRIPTION:
WHITE OAK CREEK 46.0
END DESCRIPTION:
XS GIS Cut Line= 3
      2682213.55     10037619.39      2682616.33     10037487.45
      2683560.79     10036320.76
#Sta/Elev= 30
  4311.9 1880.96  4388.8 1880.71  4509.3 1882.61  4775.8 1879.86  4804.5  1877.1
  4817.7 1872.66 4842.33 1857.35  4846.2 1854.29  4860.5 1849.33  4874.9 1847.95
  4924.5 1849.69  4967.6  1845.1  4993.4 1844.69  4996.1 1844.19  4999.4 1844.69
  5031.6 1846.46  5052.4 1854.11  5095.5 1855.62  5499.1 1857.05  5657.4 1858.78
  5749.4 1862.38    5799 1867.66  5848.6 1882.41  5906.1 1903.56    6034 1941.53
  6062.8 1946.97  6092.6    1950  6105.6 1951.82  6155.5 1958.94  6236.8 1960.56
#Mann= 8 ,-1 , 0
  4311.9     .05       0  4388.8      .1       0  4993.4     .07       0
  4999.4      .1       0  5499.1     .05       0  5657.4      .1       0
  6092.6     .16       0  6105.6      .1       0
Bank Sta=4842.33,5095.5
XS Rating Curve= 0 ,0
Exp/Cntr=0.3,0.1

Type RM Length L Ch R = 1 ,31977   ,392,392,392
BEGIN DESCRIPTION:
WHITE OAK CREEK 45.0
END DESCRIPTION:
XS GIS Cut Line= 4
      2682199.71     10037716.62      2682914.95     10037799.95
      2683664.95     10036765.22        2683658.      10036320.8
#Sta/Elev= 30
  4166.9 1879.85  4300.1 1880.57  4342.9 1880.52  4558.3 1876.33  4709.3 1866.72
    4810 1863.48  4930.6 1862.61  4951.4 1859.44  4957.6 1857.09 4957.95 1855.47
    4987  1843.9  4998.7 1842.07  5001.4 1841.57  5004.7 1842.07  5037.2  1843.6
  5066.6 1849.62  5087.5 1851.94  5158.6 1854.53  5193.2 1854.78  5241.5  1854.2
  5745.3 1855.34  5749.6  1855.4  5882.7 1858.42  6132.1 1873.81  6196.4 1885.72
  6260.5 1895.02  6376.4 1920.72  6496.5 1941.29  6526.5 1944.56  6609.4 1948.99
#Mann= 9 ,-1 , 0
  4166.9      .1       0  4300.1     .05       0  4342.9      .1       0
  4998.7     .07       0  5004.7      .1       0  5193.2     .05       0
  5241.5      .1       0  5745.3     .16       0  5749.6      .1       0
Bank Sta=4957.95,5158.6
XS Rating Curve= 0 ,0
Exp/Cntr=0.3,0.1

Type RM Length L Ch R = 1 ,31585   ,1297,1297,1297
BEGIN DESCRIPTION:
WHITE OAK CREEK 44.0
END DESCRIPTION:
XS GIS Cut Line= 3
      2682585.11     10037926.69      2683223.97     10038051.68
      2684168.42     10036419.74
#Sta/Elev= 30
  4197.8 1873.55  4252.2 1871.71  4361.9 1863.11    4488 1861.15  4518.1 1860.85
  4933.2  1858.8  4956.2 1858.84  4961.9 1858.13 4969.89 1854.37  4973.5 1847.59
  4983.4 1842.04  5001.9 1840.91  5004.7 1840.41  5007.9 1840.91  5054.4 1847.28
  5085.3 1849.76  5169.6 1851.24    5371 1852.31    5398 1852.63  5481.8 1852.86
  5620.5 1852.15  5722.5 1854.52  5856.1 1859.77  5871.8 1860.34  6204.7 1876.41
  6306.6 1879.53  6565.5 1895.09  6602.9 1897.18  6701.2 1902.43  6734.3 1904.19
#Mann= 16 ,-1 , 0
  4197.8      .1       0    4488     .05       0  4518.1      .1       0
  4933.2     .16       0  4956.2      .1       0  5001.9     .07       0
  5007.9      .1       0  5169.6     .05       0    5371     .16       0
    5398     .05       0  5481.8      .1       0  5856.1     .16       0
  5871.8      .1       0  6565.5     .05       0  6602.9      .1       0
  6701.2     .05       0
Bank Sta=4969.89,5722.5
XS Rating Curve= 0 ,0
Exp/Cntr=0.3,0.1

Type RM Length L Ch R = 1 ,30172   ,276,276,276
BEGIN DESCRIPTION:
Mapping XS 0e324681
END DESCRIPTION:
XS GIS Cut Line= 4
      2682611.85      10037996.8      2683766.35     10038226.83
      2684708.19      10037458.6      2684942.58     10036759.78
#Sta/Elev= 30
  2838.2 1870.12  2946.1 1863.15  3031.1  1861.8  3222.3 1859.94  3417.2 1859.02
  3516.9 1858.59  3864.6 1858.39  3977.9 1856.56  4075.9 1858.13  4232.5 1851.15
    4445 1851.24  4900.2 1845.04  4908.1  1844.5    4972 1839.81  4992.6 1836.13
  5021.6 1838.97    5036 1843.34  5042.4 1851.48  5050.3 1854.28  5085.5 1873.86
  5114.2 1878.86  5141.5 1886.56  5198.9 1890.62  5249.6  1891.3  5281.1 1889.65
  5307.4 1885.25  5330.9 1884.77    5402 1893.48  5478.5 1898.24  5967.9 1916.09
#Mann= 8 ,-1 , 0
  2838.2      .1       0  3031.1     .05       0  3222.3      .1       0
  3417.2     .16       0  3516.9      .1       0  4908.1     .07       0
  5042.4     .16       0  5307.4      .1       0
Bank Sta=4900.2,5036
XS Rating Curve= 0 ,0
Exp/Cntr=0.3,0.1

Type RM Length L Ch R = 1 ,29896   ,2134,2134,2134
BEGIN DESCRIPTION:
WHITE OAK CREEK 42.0
END DESCRIPTION:
XS GIS Cut Line= 5
      2683024.33     10040143.69      2683996.54      10038937.1
       2684239.6     10038277.38        2684908.     10037600.29
      2685367.37     10036837.58
#Sta/Elev= 30
  2092.6 1901.33  2202.3 1893.48  2237.5 1887.75  2387.8 1872.54  2571.8 1862.47
    2786 1855.95  3112.4 1853.08  3397.1 1855.76  3595.5 1861.07  3980.9 1845.61
  4361.2 1841.75  4410.6 1836.97  4424.8 1838.56    4453 1847.53  4474.3 1848.93
  4580.3 1850.27  4806.6 1848.11  4933.9 1845.38  5004.4 1834.27  5032.9 1837.51
    5047 1842.44  5054.1  1847.4  5061.2 1853.23  5068.2 1863.63  5089.5  1883.6
  5103.6 1892.32  5110.6 1893.72  5409.7 1897.02  5636.9 1901.07    6187 1911.58
#Mann= 5 ,-1 , 0
  2092.6      .1       0  4806.6     .07       0  5061.2      .1       0
  5409.7     .16       0  5636.9      .1       0
#XS Ineff= 1 ,-1
 3590.91 4582.39 1850.16
Permanent Ineff=
       F
Bank Sta=4806.6,5054.1
XS Rating Curve= 0 ,0
Exp/Cntr=0.3,0.1

Type RM Length L Ch R = 1 ,27762   ,1091,1091,1091
BEGIN DESCRIPTION:
WHITE OAK CREEK 41.0
END DESCRIPTION:
XS GIS Cut Line= 4
        2683033.     10040325.99      2683987.86     10039483.97
      2684482.65     10039319.04       2685272.6     10038268.68
#Sta/Elev= 30
  3485.9 1910.57  3541.4 1907.93  3817.1 1887.95  3838.9 1883.38  3894.9    1876
  4022.9 1868.19  4037.2 1865.46  4058.1 1866.08  4150.1 1860.64  4313.2 1854.53
  4490.6 1851.04  4731.6 1850.18  4938.9 1855.33  4949.4 1854.92  4959.9 1851.29
  4965.2 1844.16    4975 1839.27  4996.9 1829.48  5020.1  1829.2  5022.9  1828.7
  5026.1  1829.2  5057.3 1835.27    5118 1834.18  5160.2 1838.73  5212.9 1840.97
  5342.6 1841.29  5566.7 1843.62  6216.5 1845.98  6510.8 1851.22  6594.8 1856.64
#Mann= 7 ,-1 , 0
  3485.9     .05       0  3541.4      .1       0  5020.1     .07       0
  5026.1      .1       0  5057.3     .16       0  5342.6      .1       0
  6510.8     .16       0
Bank Sta=4975,5160.2
XS Rating Curve= 0 ,0
Exp/Cntr=0.3,0.1

Type RM Length L Ch R = 1 ,26671   ,819,819,819
BEGIN DESCRIPTION:
WHITE OAK CREEK 40.0
END DESCRIPTION:
XS GIS Cut Line= 4
       2683892.4      10041419.7      2685046.89     10039891.96
      2685107.65     10039319.04      2685637.18     10038641.94
#Sta/Elev= 30
  2644.6 1890.82  2910.4 1880.45  3080.5 1878.35  3346.7 1876.76  3409.9    1876
  3474.4 1872.21  3596.4  1871.8  3654.6 1871.99  3730.4  1869.2  3803.2 1863.72
  3930.6 1848.48  4115.7 1842.07  4323.5 1834.17  4417.1 1837.35  4502.5  1836.1
  4508.7 1833.79  4541.4 1830.57  4719.8 1832.85    4860 1834.28    4960 1835.17
  4990.1 1826.72  5017.3 1825.81    5020 1825.31  5023.3 1825.81  5111.8 1829.19
  5161.4 1829.37  5204.7 1837.29  5268.9 1843.83  5447.2 1844.74  5995.2 1854.25
#Mann= 13 ,-1 , 0
  2644.6      .1       0  3080.5     .05       0  3346.7      .1       0
  3596.4     .05       0  3654.6      .1       0  4115.7     .05       0
  4541.4      .1       0  4719.8     .05       0    4860      .1       0
  5017.3     .07       0  5023.3      .1       0  5111.8     .16       0
  5447.2      .1       0
#XS Ineff= 1 ,-1
 4156.53 4436.93 1837.92
Permanent Ineff=
       F
Bank Sta=4960,5204.7
XS Rating Curve= 0 ,0
Exp/Cntr=0.3,0.1

Type RM Length L Ch R = 1 ,25852   ,1430,1430,1430
BEGIN DESCRIPTION:
WHITE OAK CREEK 39.0
END DESCRIPTION:
XS GIS Cut Line= 4
      2683953.14     10041621.56      2685146.72     10040221.82
      2685710.95     10040091.61      2686492.13      10038648.6
#Sta/Elev= 30
  2983.9 1903.62  3043.1 1898.17  3141.9 1897.31    3277 1889.51  3566.9 1885.48
  3691.5  1885.9  4065.4 1873.67  4190.1 1865.28  4255.8 1857.06  4328.2 1853.43
  4389.6 1847.04  4445.1 1844.43    4745 1836.65  4752.7 1836.37  4808.7 1828.34
  4938.1 1829.78  4999.5 1821.25  5030.5  1824.9  5057.8 1836.13    5063 1836.75
  5530.4  1843.4  5750.5 1843.82  5764.8 1843.32  5868.9 1843.12  6068.3 1843.98
  6094.8 1843.99  6205.1 1845.57  6548.6    1849    6778 1855.61  7043.4 1867.24
#Mann= 18 ,-1 , 0
  2983.9      .1       0  3566.9     .05       0  3691.5      .1       0
  4065.4     .05       0  4190.1      .1       0  4328.2     .05       0
  4389.6      .1       0  4445.1     .05       0    4745     .07       0
    5063      .1       0  5530.4     .05       0  5750.5      .1       0
  5764.8     .05       0  5868.9      .1       0  6068.3     .05       0
  6094.8      .1       0  6205.1     .05       0    6778      .1       0
Bank Sta=4752.7,5057.8
XS Rating Curve= 0 ,0
Exp/Cntr=0.3,0.1

Type RM Length L Ch R = 1 ,24422   ,669,669,669
BEGIN DESCRIPTION:
WHITE OAK CREEK 37.0
END DESCRIPTION:
XS GIS Cut Line= 4
       2685331.2     10042923.61      2686199.23     10041534.76
       2686470.5     10039158.45      2686796.01     10037932.37
#Sta/Elev= 30
  2802.7 1898.52  3052.4 1890.98  3144.2 1889.42  3514.4  1880.4  3614.4 1878.39
  3787.7 1873.99  4461.7 1865.72  4501.9 1863.35  4713.3  1862.2  4844.1 1852.68
  4914.1 1835.17  4919.1 1835.12  4924.7 1830.79  4954.8 1823.19  4994.9 1816.97
  5208.8 1832.19  5327.3 1834.25  5713.5 1832.46  5860.7 1835.29  6041.9 1834.32
  6857.8 1849.87  7188.9 1862.76  7309.7 1870.74  7384.9 1873.03  7580.6 1891.48
  7706.3 1908.56  7736.1 1909.67  7797.5 1925.78    8027 1974.75  8100.8 1978.65
#Mann= 9 ,-1 , 0
  2802.7      .1       0  3052.4     .05       0  3144.2      .1       0
  3514.4     .05       0  3614.4      .1       0  4914.1     .07       0
  5208.8      .1       0  6041.9      .1       0  7797.5     .16       0
#XS Ineff= 1 ,-1
 5384.66 5857.95 1834.24
Permanent Ineff=
       F
Bank Sta=4924.7,5208.8
XS Rating Curve= 0 ,0
Exp/Cntr=0.3,0.1

Type RM Length L Ch R = 1 ,23753   ,1127,1127,1127
BEGIN DESCRIPTION:
WHITE OAK CREEK 36.0
END DESCRIPTION:
XS GIS Cut Line= 4
      2686286.04     10042728.34      2686915.38     10041664.96
      2686926.23      10039169.3      2686980.44     10038117.74
#Sta/Elev= 30
  3152.5 1878.16  4419.4 1865.03  4868.1 1854.98  4879.4 1854.45  4889.4 1849.92
  4919.4 1827.61  4959.4 1818.99  5006.4 1816.55  5009.1 1816.05  5012.4 1816.55
  5029.4 1821.79  5069.4 1825.22  5210.8    1826  5339.4 1828.24  5429.4 1827.86
  5449.4 1830.44  6179.4 1828.02  6599.4 1830.51  6889.4 1846.54  6909.4 1843.75
  6919.5 1848.83  6994.4 1854.94  7109.7 1865.82  7229.9  1886.9  7417.4 1912.31
  7560.3 1920.73  7613.9 1930.73  7750.6 1949.72  7810.6 1960.91  7936.8 1976.58
#Mann= 8 ,-1 , 0
  3152.5      .1       0  4868.1     .16       0  5006.4     .07       0
  5012.4     .16       0  5210.8      .1       0  6994.4     .16       0
  7417.4      .1       0  7613.9     .16       0
Bank Sta=4919.4,5339.4
XS Rating Curve= 0 ,0
Exp/Cntr=0.3,0.1

Type RM Length L Ch R = 1 ,22626   ,1594,1594,1594
BEGIN DESCRIPTION:
WHITE OAK CREEK 34.0
END DESCRIPTION:
XS GIS Cut Line= 4
      2687403.66     10041957.94      2687859.39      10040601.6
      2687360.26     10039950.55      2687121.55     10038181.91
#Sta/Elev= 30
  3290.4 1860.16  3575.6 1854.19  3646.1 1852.91  4077.7 1840.84  4642.5 1837.62
    4892 1840.61  4912.8 1837.87 4931.82 1825.68  4933.7 1820.78  4948.2 1816.14
    4995 1813.56  4997.8 1813.06    5001 1813.56  5070.6 1814.43  5112.3 1820.74
  5205.7 1818.71  5593.2 1824.71  5780.6 1822.14  6039.4 1825.05  6254.9 1828.96
  6406.2 1838.37  6507.1 1860.79  6547.5 1863.05  6628.2 1900.45    6719 1948.52
  6749.3 1959.02  6857.5 1963.47  6951.1    1960  7092.5 1960.77  7326.3 1976.47
#Mann= 7 ,-1 , 0
  3290.4     .05       0  3575.6      .1       0  3646.1     .05       0
  4642.5      .1       0    4995     .07       0    5001      .1       0
  6857.5     .16       0
Bank Sta=4931.82,5593.2
XS Rating Curve= 0 ,0
Exp/Cntr=0.3,0.1

Type RM Length L Ch R = 1 ,21032   ,1254,1254,1254
BEGIN DESCRIPTION:
WHITE OAK CREEK 30.0
END DESCRIPTION:
XS GIS Cut Line= 4
      2687588.13     10041925.37      2688228.31     10039983.11
      2688304.27     10038778.68      2689703.73     10038084.37
#Sta/Elev= 30
  2224.6 1854.94  2818.9 1839.92    3458 1834.82  3567.6 1836.38  3858.3 1834.67
  3952.4 1833.65  3974.8  1833.6  4330.6 1831.09  4575.4 1828.24  4709.9 1819.22
  4840.2 1821.18  4982.9    1809  4997.5  1807.9  5000.2  1807.4  5003.5  1807.9
  5120.7 1821.38  5179.1  1826.9  5220.9 1824.15  5768.8 1849.66  5961.2  1857.8
  6012.7 1866.97  6041.9  1880.8  6242.7 1936.51  6400.5 1962.07  6519.3 1974.48
  6601.3 1976.86  6775.9 1981.02  6927.8 1995.58    6993 1999.32  7038.7 2000.46
#Mann= 18 ,-1 , 0
  2224.6     .05       0    3458      .1       0  3567.6     .05       0
  3858.3      .1       0  3952.4     .05       0  3974.8      .1       0
  4330.6     .05       0  4575.4      .1       0  4982.9     .16       0
  4997.5     .07       0  5003.5     .16       0  5179.1      .1       0
  5768.8     .05       0  6012.7      .1       0  6242.7     .16       0
  6601.3      .1       0  6927.8     .16       0    6993      .1       0
#XS Ineff= 1 ,-1
 4622.76 4832.53 1821.94
Permanent Ineff=
       F
Bank Sta=4840.2,5120.7
XS Rating Curve= 0 ,0
Exp/Cntr=0.3,0.1

Type RM Length L Ch R = 1 ,19778   ,986,986,986
BEGIN DESCRIPTION:
WHITE OAK CREEK 29.0
END DESCRIPTION:
XS GIS Cut Line= 4
      2687772.57     10041643.28      2688792.55     10040221.82
      2689324.23     10039907.15      2690018.67     10039993.96
#Sta/Elev= 30
  2838.5 1846.74  3007.8  1840.2  3743.8 1828.24    3971 1827.09    4246 1826.91
  4397.9 1828.09    4613 1818.73  4920.3 1815.35  4969.9 1809.99  5010.2 1799.47
    5013 1798.97  5016.2 1799.47  5047.6 1802.25  5145.4 1814.66  5175.9 1832.38
  5182.4 1839.56  5210.5 1850.12  5221.9 1858.91  5277.2 1865.75  5371.4 1878.52
  5431.8 1899.03  5472.2 1905.53    5620 1915.13  5633.4 1918.66  5643.5 1918.63
  5663.6 1910.88  5683.8 1909.84  5734.2 1927.22  5791.7 1937.37  5905.7 1957.78
#Mann= 9 ,-1 , 0
  2838.5     .05       0  3743.8      .1       0    3971     .05       0
    4246      .1       0  5010.2     .07       0  5016.2      .1       0
  5047.6     .16       0  5277.2      .1       0  5791.7     .16       0
Bank Sta=4920.3,5145.4
XS Rating Curve= 0 ,0
Exp/Cntr=0.3,0.1

Type RM Length L Ch R = 1 ,18792   ,645,645,645
BEGIN DESCRIPTION:
WHITE OAK CREEK 27.0
END DESCRIPTION:
XS GIS Cut Line= 4
      2687815.98     10041947.09      2688901.06     10040970.52
       2689595.5     10040927.12      2690018.67     10040330.34
#Sta/Elev= 30
  3156.3  1850.5  4080.7 1829.93    4357 1816.54  4793.9 1810.07  4924.1 1803.87
  4991.3 1797.27    4994 1796.77  4997.3 1797.27  5025.8 1799.92  5044.4 1801.51
  5064.4 1811.66  5144.6 1827.05  5291.1 1835.01  5325.4 1835.34  5517.1 1842.84
  5638.9 1861.86    5725 1882.52  5739.8 1888.81  5775.5 1893.15  5790.3 1899.92
  5811.2 1901.55  5825.9 1907.85  5846.8 1908.69  5861.6 1913.73  5897.3 1913.95
  5912.1 1918.63  5983.4 1921.82  5998.2 1926.24  6033.9 1929.26  6043.5 1927.37
#Mann= 7 ,-1 , 0
  3156.3     .05       0  4080.7      .1       0  4991.3     .07       0
  4997.3      .1       0  5025.8     .16       0  5291.1      .1       0
  5325.4     .16       0
Bank Sta=4793.9,5064.4
XS Rating Curve= 0 ,0
Exp/Cntr=0.3,0.1

Type RM Length L Ch R = 1 ,18147   ,631,631,631
BEGIN DESCRIPTION:
WHITE OAK CREEK 26.0
END DESCRIPTION:
XS GIS Cut Line= 4
      2687772.62     10042229.19      2688901.06     10041936.23
      2689584.65     10041252.64      2690051.23      10040579.9
#Sta/Elev= 30
  3329.5 1856.53  3771.9 1845.84  4154.4 1843.32  4306.7 1843.82  4399.7 1839.93
  4530.6 1827.93  4771.1 1820.37  4827.6 1814.71    4870 1806.55  4879.5 1803.61
  4898.3 1799.43  4976.1 1797.67  4983.2 1794.73  5001.4    1794  5004.1  1793.5
  5007.4    1794  5075.1    1798  5103.4 1805.27  5117.5 1809.37  5230.7 1814.23
  5336.7 1826.52  5405.7 1830.55  5521.6 1833.47  5758.6  1824.1  5952.5 1834.06
    6003 1839.41  6095.7 1849.18  6125.4 1858.76  6176.1 1867.39  6280.8 1877.23
#Mann= 7 ,-1 , 0
  3329.5     .05       0  4154.4      .1       0  4879.5     .16       0
  5001.4     .07       0  5007.4     .16       0  5405.7      .1       0
    6003     .16       0
Bank Sta=4870,5103.4
XS Rating Curve= 0 ,0
Exp/Cntr=0.3,0.1

Type RM Length L Ch R = 1 ,17516   ,495,495,495
BEGIN DESCRIPTION:
WHITE OAK CREEK 25.0
END DESCRIPTION:
XS GIS Cut Line= 4
      2688618.17     10042546.31      2689586.91     10042103.61
      2689842.12     10041832.77      2691232.79     10041817.15
#Sta/Elev= 30
  3748.8 1844.19  4072.4 1841.23  4157.4 1841.14  4225.8 1836.96  4328.2 1826.41
  4429.6 1823.33  4768.7 1817.98  4808.6 1817.77  4864.5 1818.29  4885.6 1816.18
  4913.9 1800.44  4935.3 1793.85  4995.8 1792.73  4998.6 1792.23  5001.8 1792.73
  5048.2    1795  5069.6 1798.15  5112.1 1798.43  5126.3 1801.28  5168.8 1806.05
  5212.4 1806.56  5242.4 1799.43  5282.4 1796.96  5292.4 1794.39  5502.4 1813.69
  5662.4 1818.41  5822.4 1832.03  5981.4 1833.03  6550.3 1838.18  6576.8 1837.85
#Mann= 11 ,-1 , 0
  3748.8     .05       0  4072.4      .1       0  4157.4     .05       0
  4328.2     .16       0  4429.6      .1       0  4768.7     .05       0
  4808.6      .1       0  4995.8     .07       0  5001.8      .1       0
  5981.4     .05       0  6550.3      .1       0
#XS Ineff= 1 ,-1
 5196.31 5659.66 1806.97
Permanent Ineff=
       F
Bank Sta=4913.9,5126.3
XS Rating Curve= 0 ,0
Exp/Cntr=0.3,0.1

Type RM Length L Ch R = 1 ,17021   ,531,531,531
BEGIN DESCRIPTION:
WHITE OAK CREEK 24.0
END DESCRIPTION:
XS GIS Cut Line= 2
      2688898.58     10042677.38      2691233.52     10041861.45
#Sta/Elev= 30
    3805 1839.57  3914.7 1837.54  4018.1 1837.31  4108.7 1836.23  4186.2 1832.97
  4260.6 1824.06  4304.3 1821.35  4478.9 1817.59  4641.7 1816.42  4676.6 1814.48
  4798.3 1812.89  4906.5 1798.61  4959.5 1793.16  4998.9 1785.61  5001.6 1785.11
  5004.9 1785.61  5018.8 1787.68  5046.7 1789.38  5072.4 1794.35  5086.6 1793.78
  5108.8 1790.36  5160.3 1798.61  5227.6 1808.57  5253.4 1816.24  5284.4  1818.5
  5408.6  1820.8  5658.6 1831.76  5803.7 1831.99  6248.4 1836.65  6278.4 1836.44
#Mann= 13 ,-1 , 0
    3805     .05       0  3914.7      .1       0  4018.1     .05       0
  4108.7     .16       0  4304.3      .1       0  4478.9     .05       0
  4676.6      .1       0  4998.9     .07       0  5004.9      .1       0
  5018.8     .05       0  5086.6      .1       0  5803.7     .05       0
  6248.4      .1       0
Bank Sta=4906.5,5160.3
XS Rating Curve= 0 ,0
Exp/Cntr=0.3,0.1

Type RM Length L Ch R = 1 ,16490   ,536,536,536
BEGIN DESCRIPTION:
WHITE OAK CREEK 23.0
END DESCRIPTION:
XS GIS Cut Line= 3
      2688816.08     10042950.83      2690044.38     10042877.04
      2691472.32     10042056.74
#Sta/Elev= 30
  3528.6 1842.98  3798.4 1838.07  3996.6 1834.48  4095.7 1836.58  4272.1 1835.39
  4492.7 1830.68  4542.8 1825.74  4602.9 1811.53    4633 1807.19  4713.1 1803.94
    4800 1803.07  4844.6 1798.69    4859 1795.47  4874.8 1791.57  4998.2 1783.22
  5014.2 1785.03  5035.8 1793.19  5051.6 1795.88  5063.7 1798.23  5094.8 1803.48
  5153.7 1809.16  5202.6 1816.96  5255.8 1822.49  5395.2 1824.57  5540.5 1826.52
  5797.8 1824.63  5928.6 1827.09  6076.7 1833.28  6287.4 1836.37  6405.9 1840.25
#Mann= 10 ,-1 , 0
  3528.6      .1       0  3798.4     .05       0  3996.6      .1       0
  4095.7     .16       0  4272.1      .1       0  4492.7      .1       0
  4844.6     .09       0  5063.7      .1       0  5395.2      .1       0
  6287.4     .05       0
Bank Sta=4859,5051.6
XS Rating Curve= 0 ,0
Exp/Cntr=0.3,0.1

Type RM Length L Ch R = 1 ,15954   ,588,588,588
BEGIN DESCRIPTION:
WHITE OAK CREEK 22.0
END DESCRIPTION:
XS GIS Cut Line= 3
      2688781.37     10043189.55      2690213.65     10043363.16
      2691723.78     10042382.44
#Sta/Elev= 30
  3383.1 1841.77  3676.5 1839.39  3882.1  1839.1  4118.6 1836.86  4326.1 1834.77
  4364.6  1833.9  4447.9 1832.73  4528.5 1827.95    4599 1816.66  4623.6 1811.37
  4649.4 1802.04  4669.5 1799.06  4887.2 1796.43  4944.5 1793.39  4974.7 1790.99
  4986.7 1784.27  5001.6  1781.3  5068.4 1784.35  5089.5 1788.32  5140.9  1793.6
  5153.5 1794.86  5276.7 1803.75  5320.5  1802.9  5385.4 1806.08  5566.7 1809.22
  5608.9 1816.76  5660.3 1819.11  5747.9 1819.55  6007.6 1830.41  6626.5 1848.65
#Mann= 8 ,-1 , 0
  3383.1      .1       0  3676.5     .05       0  3882.1      .1       0
  4118.6     .16       0  4326.1      .1       0  4364.6     .16       0
  4887.2     .09       0  5153.5      .1       0
Bank Sta=4944.5,5140.9
XS Rating Curve= 0 ,0
Exp/Cntr=0.3,0.1

Type RM Length L Ch R = 1 ,15366   ,1197,1197,1197
BEGIN DESCRIPTION:
WHITE OAK CREEK 21.0
END DESCRIPTION:
XS GIS Cut Line= 6
      2689752.51     10045507.66      2690403.54     10044382.69
       2690445.2     10043986.85      2690773.33     10043653.52
      2690778.54      10043330.6       2691823.5     10042498.79
#Sta/Elev= 30
  2735.4 1841.21  3496.3 1819.59  3802.9 1802.75  4094.4 1795.48  4124.6 1798.07
  4144.7 1791.79  4164.8 1797.27  4265.4 1806.25  4315.7 1801.45  4320.9 1794.89
  4325.9 1795.89  4345.8 1785.72  4365.9 1790.82  4444.8 1792.88  4671.1 1791.71
  4678.1 1791.34  4819.5 1784.04    4862 1784.16  4897.3 1789.51  4940.7 1788.23
  5000.5 1778.56  5030.7 1790.12  5080.7 1791.79  5110.7 1798.06  5150.7 1800.09
  5546.8 1805.74  5825.9 1827.79  5956.9 1832.91  6317.7 1850.61  6559.5  1854.6
#Mann= 6 ,-1 , 0
  2735.4      .1       0  4265.4     .16       0  4678.1     .09       0
  5080.7      .1       0  5546.8     .16       0  5956.9      .1       0
#XS Ineff= 2 ,-1
  3514.2 4255.68 1806.18 4281.25 4630.68 1793.29
Permanent Ineff=
       F       F
Bank Sta=4671.1,5080.7
XS Rating Curve= 0 ,0
Exp/Cntr=0.3,0.1

Type RM Length L Ch R = 1 ,14169   ,520,520,520
BEGIN DESCRIPTION:
WHITE OAK CREEK 19.0
END DESCRIPTION:
XS GIS Cut Line= 4
      2689887.88     10045523.34      2690976.45     10044611.85
      2691601.45     10044497.27      2692601.46     10042908.72
#Sta/Elev= 30
    3277 1839.21  3519.1 1832.47    3711 1825.52  3759.7 1824.07  3942.7 1820.39
  4107.7  1822.5  4228.9 1821.27  4317.9 1813.92  4399.3  1797.8  4575.1 1793.61
  4878.6 1792.04  4922.5 1788.93  4942.6 1776.11  5166.5  1783.9  5412.1 1788.01
  5631.1 1785.56  5667.2 1789.34  5898.4 1796.27  5956.1  1813.9  6007.9 1812.47
  6013.8 1814.72  6029.1 1812.22  6065.6 1813.53  6196.3 1837.14  6333.9  1845.2
  6378.2 1846.69    6559  1850.8  6686.9 1853.18  7063.7  1859.1  7209.3 1862.28
#Mann= 16 ,-1 , 0
    3277      .1       0  3519.1      .1       0    3711     .05       0
  3759.7      .1       0  3942.7     .05       0  4107.7      .1       0
  4317.9     .05       0  4575.1      .1       0  4922.5     .09       0
  5631.1     .05       0  6007.9      .1       0  6333.9     .05       0
  6378.2      .1       0    6559     .05       0  6686.9      .1       0
  7063.7     .16       0
#XS Ineff= 1 ,-1
 5411.93 5775.57 1788.84
Permanent Ineff=
       F
Bank Sta=4922.5,5667.2
XS Rating Curve= 0 ,0
Exp/Cntr=0.3,0.1

Type RM Length L Ch R = 1 ,13649   ,901,901,901
BEGIN DESCRIPTION:
WHITE OAK CREEK 18.0
END DESCRIPTION:
XS GIS Cut Line= 3
      2690721.42     10045905.17      2691567.77     10045047.96
      2692673.15     10043108.13
#Sta/Elev= 30
  3534.8 1830.32  3577.8    1829  3636.4 1827.93  3869.5 1823.01  4087.7 1807.47
  4214.5 1800.04  4375.2 1789.54  4617.3 1788.59  4917.6 1790.65    4940 1791.37
  4955.1 1784.25  4970.9 1774.96    4998 1772.72  5101.1 1780.93  5293.6 1784.92
  5439.1 1781.49  5476.6 1786.15  5535.7 1797.71    5563 1809.16  5600.5 1816.23
  5748.3 1817.83  6003.9 1826.99    6122 1837.71  6411.2 1849.88  6445.4 1852.08
  6534.4  1855.9  6609.9 1859.55  6859.3 1865.03  6877.2 1864.92  6972.1  1864.5
#Mann= 16 ,-1 , 0
  3534.8      .1       0  3577.8     .05       0  3636.4      .1       0
  3869.5     .05       0  4087.7      .1       0  4214.5     .05       0
  4617.3      .1       0  4917.6     .09       0  5535.7     .16       0
  5748.3      .1       0  6411.2     .05       0  6445.4      .1       0
  6534.4     .05       0  6609.9      .1       0  6859.3     .16       0
  6877.2     .05       0
#XS Ineff= 1 ,-1
 4247.73 4941.76 1791.54
Permanent Ineff=
       F
Bank Sta=4955.1,5476.6
XS Rating Curve= 0 ,0
Exp/Cntr=0.3,0.1

Type RM Length L Ch R = 1 ,12748   ,914,914,914
BEGIN DESCRIPTION:
WHITE OAK CREEK 16.0
END DESCRIPTION:
XS GIS Cut Line= 4
      2691177.13     10046176.46       2692001.8     10045275.83
      2692566.04     10045156.47      2693704.42     10043573.58
#Sta/Elev= 30
  3571.5 1827.34  3709.2 1820.84  3835.9 1809.56  4027.7 1805.93  4381.2 1800.68
  4643.3 1779.31  4693.2 1783.62  4777.7 1785.89  4830.7 1782.95  4893.8 1781.31
  4952.8 1776.55  4980.4 1769.82  4983.2 1769.32  4986.4 1769.82  5024.8 1771.62
    5055 1786.12  5120.9  1789.2  5709.5 1785.68  6290.1 1792.75  6518.5 1799.39
  6577.4 1807.53  6749.2 1813.04  6770.1 1821.36  6841.3 1820.79  6900.1 1834.41
  6935.8 1836.45  6977.6  1850.4  7005.1 1852.57  7179.9 1867.02  7319.1 1872.05
#Mann= 12 ,-1 , 0
  3571.5     .05       0  3709.2      .1       0  3835.9     .05       0
  4027.7      .1       0  4693.2     .16       0  4830.7      .1       0
  4893.8     .16       0  4980.4     .07       0  4986.4     .16       0
  5120.9      .1       0  7005.1     .05       0  7179.9      .1       0
#XS Ineff= 1 ,-1
 4379.55 4761.36 1787.03
Permanent Ineff=
       F
Bank Sta=4777.7,5055
XS Rating Curve= 0 ,0
Exp/Cntr=0.3,0.1

Type RM Length L Ch R = 1 ,11834   ,3011,3011,3011
BEGIN DESCRIPTION:
WHITE OAK CREEK 15.0
END DESCRIPTION:
XS GIS Cut Line= 3
      2691795.65     10046675.55      2692696.25     10045644.75
      2693857.28     10043843.52
#Sta/Elev= 30
  4179.4 1822.91  4611.6 1811.55  4891.3 1807.07    4934  1795.8  4948.3  1784.1
  4969.2 1769.03    4988 1763.57  4990.8 1763.07    4994 1763.57  5032.8 1774.85
  5097.3 1771.46  5111.3 1775.59  5175.2 1781.17  5302.3  1783.9  5585.5 1785.27
  6432.4 1779.91  6780.3 1783.67    6977 1790.75  7034.4 1797.95  7076.6 1797.38
  7155.6 1807.22    7318 1820.29  7345.9 1823.94  7388.2 1836.01  7445.6 1840.79
  7493.7    1850  7554.5  1860.6  7648.3 1859.19  7688.6 1862.03  7691.2 1862.03
#Mann= 7 ,-1 , 0
  4179.4     .05       0  4611.6      .1       0    4988     .07       0
    4994      .1       0    7318     .16       0  7493.7      .1       0
  7688.6     .05       0
Bank Sta=4948.3,5302.3
XS Rating Curve= 0 ,0
Exp/Cntr=0.3,0.1

Type RM Length L Ch R = 1 ,8823    ,1090,1090,1090
BEGIN DESCRIPTION:
WHITE OAK CREEK 14.0
END DESCRIPTION:
XS GIS Cut Line= 3
      2692273.07     10046729.82      2694095.99     10045536.25
      2694985.75     10043973.74
#Sta/Elev= 30
  2133.3 1820.66  2619.9 1809.07  2622.6 1808.98  2864.2 1804.08    3298 1805.71
  3348.4 1805.88  3469.8 1801.95  3578.8 1797.47  3666.2  1784.2  3759.7 1780.13
  4683.4 1776.17  4756.3 1773.47  4932.2 1768.32  4969.6 1763.68  4988.3 1757.09
    4991 1756.59  4994.3 1757.09  5028.6 1760.48    5072 1776.45  5115.2 1800.22
  5165.3 1803.94  5319.8 1820.11  5357.3 1827.83    5497 1838.85    5680 1846.28
  5771.8 1844.18  5868.8 1840.37  5953.2 1848.23  5981.2 1852.96  6110.3 1856.86
#Mann= 12 ,-1 , 0
  2133.3     .05       0  2619.9      .1       0  2622.6     .05       0
    3298      .1       0  3348.4     .05       0  3469.8      .1       0
  4756.3     .16       0  4988.3     .07       0  4994.3     .16       0
  5165.3      .1       0  5771.8     .05       0  5953.2      .1       0
Bank Sta=4683.4,5072
XS Rating Curve= 0 ,0
Exp/Cntr=0.3,0.1

Type RM Length L Ch R = 1 ,7733    ,505,505,505
BEGIN DESCRIPTION:
WHITE OAK CREEK 12.0
END DESCRIPTION:
XS GIS Cut Line= 4
      2692457.54     10046773.22      2694388.95     10045905.17
      2695593.38     10045850.92       2696450.6     10045113.06
#Sta/Elev= 30
  2362.7  1817.1  2497.2 1815.26  2588.9  1812.3  2628.2 1810.76  2835.1 1805.72
  3376.9  1796.6  3566.6 1786.84  3930.4 1781.86  4063.1  1775.6  4426.5 1775.67
  4624.1 1771.83  4800.1 1769.69  4825.8 1762.29  4960.2 1762.78  5017.3 1756.75
    5020 1756.25  5023.3 1756.75  5080.3 1764.86  5100.4 1771.57  5140.4 1779.16
    5200 1783.58  5520.8 1797.63  5685.9 1797.35  5832.6  1802.1  6032.1 1808.37
  6439.2 1825.36    6595 1839.91  6701.4 1838.34  6715.7 1834.62  6816.9 1835.97
#Mann= 12 ,-1 , 0
  2362.7     .05       0  2497.2      .1       0  2588.9     .05       0
  2628.2      .1       0  2835.1     .05       0  3376.9      .1       0
  4825.8     .16       0  5017.3     .07       0  5023.3     .16       0
    5200      .1       0  5832.6     .16       0  6032.1      .1       0
Bank Sta=4624.1,5100.4
XS Rating Curve= 0 ,0
Exp/Cntr=0.3,0.1

Type RM Length L Ch R = 1 ,7228    ,692,692,692
BEGIN DESCRIPTION:
WHITE OAK CREEK 11.0
END DESCRIPTION:
XS GIS Cut Line= 4
      2692566.01     10046946.85      2694237.04     10046263.24
      2695289.56     10046458.55      2696461.44     10045926.87
#Sta/Elev= 30
  2638.1 1819.65  2949.5 1814.33  3068.2 1809.93    3218 1804.71  3418.4 1797.45
  3558.7 1790.74  3715.9    1784  4191.3 1774.29    4472 1774.08  4678.9 1769.46
    4862 1763.91    4923 1758.01  4967.9 1758.14  4991.2 1751.19    4994 1750.69
  4997.2 1751.19  5034.9 1759.46  5078.6 1763.55  5095.9 1770.06  5125.4 1776.94
  5146.8 1784.39  5177.3 1786.93  5248.5 1776.54  5529.4 1778.56    5973 1787.47
  6226.6 1799.64  6424.3 1813.93  6523.1 1816.99  6696.4 1830.75  6800.9 1832.54
#Mann= 12 ,-1 , 0
  2638.1     .05       0  2949.5      .1       0  3068.2     .05       0
    3218      .1       0  3418.4     .05       0  3558.7      .1       0
    4862     .16       0  4991.2     .07       0  4997.2     .16       0
  5125.4      .1       0  5529.4     .05       0    5973      .1       0
Bank Sta=4678.9,5095.9
XS Rating Curve= 0 ,0
Exp/Cntr=0.3,0.1

Type RM Length L Ch R = 1 ,6536    ,1080,1080,1080
BEGIN DESCRIPTION:
WHITE OAK CREEK 10.0
END DESCRIPTION:
XS GIS Cut Line= 4
      2692750.47     10047304.93      2693727.06     10046784.08
      2694898.94      10047087.9      2696101.73      10046307.7
#Sta/Elev= 30
  3085.9 1822.53  3429.8 1817.79  3563.5 1814.39    3763 1804.96  3772.4 1804.48
  3877.5 1799.39    3992 1786.94    4251 1776.61  4514.4 1771.79  4586.7 1767.53
  4638.4 1768.65  4727.7 1766.18  4803.7 1763.99  4893.9 1756.99  4948.3 1756.59
  4986.6 1749.32  4989.4 1748.82  4992.6 1749.32  5041.3 1753.24  5052.4 1757.57
 5065.91 1766.36  5072.3 1770.07  5082.6 1772.08  5100.6 1772.29    5245 1771.61
  5414.4 1767.97    5895 1772.77  6359.8 1780.46  6563.8  1787.7    6837 1806.12
#Mann= 13 ,-1 , 0
  3085.9     .05       0  3429.8      .1       0  3563.5     .05       0
    3763     .16       0  3772.4      .1       0  3877.5     .16       0
    3992      .1       0  4893.9     .16       0  4986.6     .07       0
  4992.6     .16       0  5100.6      .1       0    5895     .05       0
  6563.8      .1       0
Bank Sta=4727.7,5065.91
XS Rating Curve= 0 ,0
Exp/Cntr=0.3,0.1

Type RM Length L Ch R = 1 ,5456    ,465,465,465
BEGIN DESCRIPTION:
WHITE OAK CREEK 8.0
END DESCRIPTION:
XS GIS Cut Line= 4
      2693889.83     10048248.92      2694367.25     10048151.26
      2695018.29     10047424.27      2696134.72     10046481.26
#Sta/Elev= 30
  4279.4 1810.36  4481.1 1808.21  4540.3 1808.05  4578.9 1806.95  4725.7 1805.22
  4801.5 1801.86  4885.9 1799.96  4900.1 1797.18  4914.3 1790.88  4921.8 1784.98
  4942.8 1761.81    4957 1752.48  4971.2 1747.27  4996.6 1745.29  4999.3 1744.79
  5002.6 1745.29    5028 1747.05  5048.9 1751.78  5069.1 1751.81  5197.7 1762.17
  5289.2 1765.74  5488.3 1768.06  5771.1 1765.87  6136.1 1767.91  6651.3 1776.69
  6743.6 1778.98  6798.9 1782.26  6867.6 1784.79  6920.2 1786.92    7204  1802.9
#Mann= 12 ,-1 , 0
  4279.4     .05       0  4481.1      .1       0  4540.3     .05       0
  4578.9      .1       0  4996.6     .07       0  5002.6      .1       0
  5069.1     .16       0  5289.2      .1       0  6136.1     .05       0
  6798.9      .1       0  6867.6     .05       0  6920.2      .1       0
Bank Sta=4942.8,5197.7
XS Rating Curve= 0 ,0
Exp/Cntr=0.3,0.1

Type RM Length L Ch R = 1 ,4991    ,652,652,652
BEGIN DESCRIPTION:
WHITE OAK CREEK 7.0
END DESCRIPTION:
XS GIS Cut Line= 4
       2694117.7     10048878.25      2694812.13     10048389.98
       2695126.8     10047684.68      2696417.09     10046567.88
#Sta/Elev= 30
  4026.8 1818.01  4087.5 1817.15  4235.9 1813.44  4339.5  1811.7  4500.5 1807.52
  4569.2 1805.59  4661.5 1801.01  4719.9  1790.7  4799.4 1783.07  4901.2 1769.64
  4906.7 1771.74  4924.5 1766.18  4929.9  1769.4  4947.7 1764.88  4953.2 1766.55
  4959.2 1759.88  4976.4  1746.9  4996.6 1745.11  4999.4 1744.61  5002.6 1745.11
  5080.2 1750.26  5099.6 1754.29  5173.1 1760.37  5246.3 1762.92  5911.7 1764.64
  6387.4 1771.12  6732.1 1788.25  6949.7 1795.82    7167 1804.68  7354.5 1815.15
#Mann= 16 ,-1 , 0
  4026.8      .1       0  4087.5     .05       0  4235.9      .1       0
  4339.5     .05       0  4500.5      .1       0  4569.2     .05       0
  4661.5     .16       0  4799.4      .1       0  4996.6     .07       0
  5002.6      .1       0  5099.6     .16       0  5246.3      .1       0
  5911.7     .05       0  6732.1      .1       0  6949.7     .05       0
    7167      .1       0
Bank Sta=4959.2,5173.1
XS Rating Curve= 0 ,0
Exp/Cntr=0.3,0.1

Type RM Length L Ch R = 1 ,4339    ,701,701,701
BEGIN DESCRIPTION:
WHITE OAK CREEK 6.0
END DESCRIPTION:
XS GIS Cut Line= 4
      2694519.15     10049062.73      2695463.17     10048596.14
      2695517.43      10047988.5      2696547.67     10046697.99
#Sta/Elev= 30
  3588.8 1811.33  3614.8  1810.7  3758.8 1805.89    3893 1799.97  3982.8 1789.55
  4127.2  1785.7  4179.1 1782.89  4235.2 1772.64    4280 1770.36  4498.9 1764.35
  4798.4 1761.25  4865.1 1761.76  4915.3 1758.58  4935.4 1756.87  4975.6    1746
  5022.8 1744.89  5025.5 1744.39  5028.8 1744.89  5065.9 1749.57  5136.2 1751.85
  5196.4 1758.64  5251.8 1762.45  5341.4 1761.09  5391.1 1759.19  5526.7 1763.39
  5757.3 1774.41  5910.6 1784.83  6160.3 1789.09  6529.5 1796.01  6903.2 1813.64
#Mann= 10 ,-1 , 0
  3588.8      .1       0  3614.8     .05       0  3758.8      .1       0
  4127.2     .05       0  4798.4      .1       0  5022.8     .07       0
  5028.8      .1       0  5341.4     .05       0  5757.3      .1       0
  6160.3     .05       0
Bank Sta=4915.3,5196.4
XS Rating Curve= 0 ,0
Exp/Cntr=0.3,0.1

Type RM Length L Ch R = 1 ,3638    ,966,966,966
BEGIN DESCRIPTION:
WHITE OAK CREEK 5.0
END DESCRIPTION:
XS GIS Cut Line= 4
      2694779.56     10049333.99      2695539.13     10049116.98
      2696374.63      10047988.5      2696645.91     10046784.04
#Sta/Elev= 30
  3349.5 1808.04  3396.1 1806.69  3419.2 1806.27  3713.6 1799.53  3972.4 1794.86
  4019.6 1792.01  4154.1  1786.8  4248.4 1781.43    4263 1774.42  4292.3 1766.77
  4327.8 1761.35  4582.7 1758.87  4819.9 1756.68  4938.4  1751.8  4991.4 1741.11
  5023.9 1740.37  5026.7 1739.87  5029.9 1740.37  5070.8 1748.72 5086.36 1757.03
    5100 1762.11    5114 1763.98  5209.3  1764.5  5527.8 1771.03  5641.2  1775.8
  5794.5 1781.38  5937.4 1782.14    5972 1782.21  6398.6 1795.62  6778.2 1813.78
#Mann= 15 ,-1 , 0
  3349.5     .16       0  3396.1      .1       0  3419.2     .05       0
  3713.6      .1       0  4019.6     .05       0  4154.1      .1       0
  4582.7     .05       0  4819.9     .16       0  4938.4      .1       0
  5023.9     .07       0  5029.9      .1       0  5209.3      .1       0
  5641.2     .05       0  5937.4      .1       0    5972     .05       0
Bank Sta=4819.9,5086.36
XS Rating Curve= 0 ,0
Exp/Cntr=0.3,0.1
