--- NORTH GRAPE CREEK.prj (project) ---

Proj Title=NORTH GRAPE CREEK Base Level Engineering
Current Plan=p01
Default Exp/Contr=0.3,0.1
English Units
Geom File=g01
Flow File=f01
Plan File=p01
Y Axis Title=Elevation
X Axis Title(PF)=Main Channel Distance
X Axis Title(XS)=Station
BEGIN DESCRIPTION:
NORTH GRAPE CREEK
END DESCRIPTION:
DSS Export Rating Curves= 0
DSS Export Rating Curve Sorted= 0
DSS Export Volume Flow Curves= 0
DXF OffsetX= 0
DXF OffsetY= 0
DXF ScaleX= 1
DXF ScaleY= 10

--- NORTH GRAPE CREEK.p01 (plan) ---

Plan Title=Multiple Run
Short Identifier=Multiple
Geom File=g01
Flow File=f01
Subcritical Flow
K Sum by GR= 0
Std Step Tol= 0.01
Critical Tol= 0.01
Num of Std Step Trials= 20
Max Error Tol= 0.3
Flow Tol Ratio= 0.001
Split Flow NTrial= 30
Split Flow Tol= 0.02
Split Flow Ratio= 0.02
Log Output Level= 0
Friction Slope Method= 1
Unsteady Friction Slope Method= 2
Unsteady Bridges Friction Slope Method= 1
Parabolic Critical Depth
Global Vel Dist=  1 , 1 , 1
Global Log Level= 0
CheckData=True
Encroach Param= -1, 0, 0, 0
BEGIN DESCRIPTION:
Multiple Run
END DESCRIPTION:

--- NORTH GRAPE CREEK.f01 (steady flow) ---

Flow Title=Multiple
Program Version=4.10
Number of Profiles= 7
Profile Names=10-year,25-year,50-year,1pct_min,100-year,1pct_plu,500-year
River Rch & RM=NORTH GRAPE CREE,Reach-1         ,138404
     717    1022    1281    1177    1592    2153    2464
River Rch & RM=NORTH GRAPE CREE,Reach-1         ,137007
    1088    1580    2007    1863    2520    3408    3989
River Rch & RM=NORTH GRAPE CREE,Reach-1         ,130010
    1449    2134    2735    2560    3463    4683    5574
River Rch & RM=NORTH GRAPE CREE,Reach-1         ,123970
    2344    3523    4579    4339    5869    7937    9684
River Rch & RM=NORTH GRAPE CREE,Reach-1         ,117462
    2425    3648    4744    4497    6082    8225   10044
River Rch & RM=NORTH GRAPE CREE,Reach-1         ,116686
    2425    3648    4744    4497    6082    8225   10044
River Rch & RM=NORTH GRAPE CREE,Reach-1         ,116116
    2997    4546    5944    5663    7658   10357   12771
River Rch & RM=NORTH GRAPE CREE,Reach-1         ,114829
    3470    5290    6943    6634    8972   12134   15057
River Rch & RM=NORTH GRAPE CREE,Reach-1         ,113468
    3470    5290    6943    6634    8972   12134   15057
River Rch & RM=NORTH GRAPE CREE,Reach-1         ,111580
    3470    5290    6943    6634    8972   12134   15057
River Rch & RM=NORTH GRAPE CREE,Reach-1         ,111078
    4035    6174    8121    7775   10515   14220   17708
River Rch & RM=NORTH GRAPE CREE,Reach-1         ,104302
    4185    6401    8419    8058   10897   14737   18342
River Rch & RM=NORTH GRAPE CREE,Reach-1         ,99341
    4232    6456    8475    8093   10945   14802   18341
River Rch & RM=NORTH GRAPE CREE,Reach-1         ,88740
    4466    6820    8960    8561   11578   15658   19423
River Rch & RM=NORTH GRAPE CREE,Reach-1         ,83538
    4498    6864    9010    8603   11635   15735   19489
River Rch & RM=NORTH GRAPE CREE,Reach-1         ,76382
    9212   14321   19047   18397   24879   33647   42621
River Rch & RM=NORTH GRAPE CREE,Reach-1         ,75546
    9212   14321   19047   18397   24879   33647   42621
River Rch & RM=NORTH GRAPE CREE,Reach-1         ,71484
   10563   16472   21957   21251   28740   38868   49429
River Rch & RM=NORTH GRAPE CREE,Reach-1         ,70442
   11003   17190   22945   22236   30072   40669   51851
River Rch & RM=NORTH GRAPE CREE,Reach-1         ,68420
   11003   17190   22945   22236   30072   40669   51851
River Rch & RM=NORTH GRAPE CREE,Reach-1         ,63901
   11141   17414   23251   22540   30483   41225   52593
River Rch & RM=NORTH GRAPE CREE,Reach-1         ,60356
   11932   18685   24982   24250   32795   44352   56723
River Rch & RM=NORTH GRAPE CREE,Reach-1         ,56881
   12404   19445   26017   25272   34178   46222   59194
River Rch & RM=NORTH GRAPE CREE,Reach-1         ,52740
   12770   20022   26795   26031   35203   47609   60982
River Rch & RM=NORTH GRAPE CREE,Reach-1         ,47807
   12923   20255   27100   26320   35595   48137   61625
River Rch & RM=NORTH GRAPE CREE,Reach-1         ,39599
   13272   20814   27859   27067   36604   49503   63416
River Rch & RM=NORTH GRAPE CREE,Reach-1         ,35251
   13325   20888   27950   27147   36713   49650   63565
River Rch & RM=NORTH GRAPE CREE,Reach-1         ,30688
   14136   22177   29692   28853   39021   52771   67622
River Rch & RM=NORTH GRAPE CREE,Reach-1         ,29725
   14136   22177   29692   28853   39021   52771   67622
River Rch & RM=NORTH GRAPE CREE,Reach-1         ,23748
   14037   21989   29411   28551   38611   52217   66772
River Rch & RM=NORTH GRAPE CREE,Reach-1         ,14917
   14503   22716   30381   29488   39880   53933   68942
River Rch & RM=NORTH GRAPE CREE,Reach-1         ,10569
   14982   23455   31359   30424   41145   55644   71067
Boundary for River Rch & Prof#=NORTH GRAPE CREE,Reach-1         , 1
Up Type= 0
Dn Type= 3
Dn Slope=0.0016
Boundary for River Rch & Prof#=NORTH GRAPE CREE,Reach-1         , 2
Up Type= 0
Dn Type= 3
Dn Slope=0.0016
Boundary for River Rch & Prof#=NORTH GRAPE CREE,Reach-1         , 3
Up Type= 0
Dn Type= 3
Dn Slope=0.0016
Boundary for River Rch & Prof#=NORTH GRAPE CREE,Reach-1         , 4
Up Type= 0
Dn Type= 3
Dn Slope=0.0016
Boundary for River Rch & Prof#=NORTH GRAPE CREE,Reach-1         , 5
Up Type= 0
Dn Type= 3
Dn Slope=0.0016
Boundary for River Rch & Prof#=NORTH GRAPE CREE,Reach-1         , 6
Up Type= 0
Dn Type= 3
Dn Slope=0.0016
Boundary for River Rch & Prof#=NORTH GRAPE CREE,Reach-1         , 7
Up Type= 0
Dn Type= 3
Dn Slope=0.0016
DSS Import GetInterval= 0
DSS Import GetPeak= 0
DSS Import FillOption= 0

--- NORTH GRAPE CREEK.g01 (geometry) ---

Geom Title=Existing Conditions
Program Version=4.10

River Reach=NORTH GRAPE CREE,Reach-1
Reach XY= 30
      2795448.47     10093183.73      2798785.11     10094525.49
      2805025.54     10086696.42      2807065.45     10089779.25
      2812157.11     10090357.03       2813378.4     10092757.81
      2815644.67     10091373.54      2816224.29     10093021.76
      2825664.12     10093319.16      2826026.29     10096170.39
      2827925.83     10096805.12      2827359.33     10099070.42
      2829535.12     10099531.58      2830063.09     10098665.37
      2833779.05     10100632.48      2842527.07     10098772.82
      2847379.51     10092314.82      2849744.79     10091047.29
      2858098.42     10093458.77      2857683.93     10096198.11
      2858709.96     10097590.13      2868168.47     10098543.73
      2869387.18     10097511.58      2868058.98      10093616.7
      2873853.22     10095073.13      2874158.76     10093187.57
      2876226.04      10092999.2      2879541.41     10090375.72
      2875652.83     10087802.56      2877644.86     10085120.76

Type RM Length L Ch R = 1 ,138404  ,652,652,652
BEGIN DESCRIPTION:
NORTH GRAPE CREEK 188.0
END DESCRIPTION:
XS GIS Cut Line= 2
      2795301.05     10093703.96      2796124.62     10093140.47
#Sta/Elev= 30
  4599.8 1919.35  4742.1 1908.89  4764.3 1905.77  4770.4 1905.41  4785.3 1902.93
  4806.3 1901.02  4821.2 1898.96  4836.1 1898.09    4851 1897.78    4893  1898.8
  4979.7 1897.64  4997.6 1895.69  5000.4 1895.19  5003.6 1895.69  5021.6 1897.18
    5045 1896.73  5057.5 1898.22  5066.3  1900.6  5081.2 1903.31  5093.5 1905.08
  5108.3 1906.24    5180  1907.9  5296.6 1913.54  5347.3 1914.68  5374.4 1916.76
    5455 1920.02  5461.1 1920.84  5496.9 1922.75  5562.7 1925.37  5597.7 1927.31
#Mann= 3 ,-1 , 0
  4599.8     .16       0  4997.6     .07       0  5003.6     .16       0
Bank Sta=4979.7,5057.5
XS Rating Curve= 0 ,0
Exp/Cntr=0.3,0.1

Type RM Length L Ch R = 1 ,137752  ,745,745,745
BEGIN DESCRIPTION:
NORTH GRAPE CREEK 187.0
END DESCRIPTION:
XS GIS Cut Line= 2
      2795726.46     10094294.18      2796264.02      10093643.9
#Sta/Elev= 30
  4652.8    1909  4768.7  1907.2  4789.5 1906.55  4810.3 1906.43  4818.2 1906.89
    4861 1905.74  4874.1 1904.61    4882 1904.49  4901.7 1902.12  4960.1 1896.26
  4966.6 1894.64  4974.5 1891.94    4981 1888.13  4988.8 1885.59  4995.3 1884.57
  5000.1 1884.54  5002.9 1884.04  5006.1 1884.54  5009.6  1885.3  5016.7 1887.78
  5030.5 1890.85  5081.3 1893.56  5105.3 1894.25  5172.4 1894.09  5272.8 1896.31
  5307.9 1898.32  5336.6 1901.85  5365.3 1904.49  5414.8 1906.71  5496.5 1909.11
#Mann= 7 ,-1 , 0
  4652.8     .16       0  4768.7      .1       0  4901.7     .16       0
  5000.1     .07       0  5006.1     .16       0  5105.3      .1       0
  5414.8     .16       0
Bank Sta=4974.5,5030.5
XS Rating Curve= 0 ,0
Exp/Cntr=0.3,0.1

Type RM Length L Ch R = 1 ,137007  ,413,413,413
BEGIN DESCRIPTION:
NORTH GRAPE CREEK 186.0
END DESCRIPTION:
XS GIS Cut Line= 2
      2796308.06     10094571.96      2796941.73     10093851.48
#Sta/Elev= 30
  4499.6 1899.33    4541 1896.17  4583.7 1894.47  4720.7 1892.19  4767.7 1891.09
  4831.3 1887.11    4910 1885.72  4951.8 1883.24  4959.4 1883.79    4966 1883.25
  4973.6 1881.93  4987.8  1877.6  4999.1 1876.34  5001.8 1875.84  5005.1 1876.34
  5008.7 1876.38  5016.3  1879.1  5022.9 1883.88  5026.9 1887.09  5029.9  1889.5
  5058.1 1892.72  5079.9 1894.03  5094.1 1896.44  5143.4 1901.83  5186.1  1904.1
  5284.8 1906.92  5335.9 1909.39  5380.1 1910.78  5427.1  1912.7  5459.1 1913.19
#Mann= 7 ,-1 , 0
  4499.6     .16       0  4720.7      .1       0  4999.1     .07       0
  5005.1      .1       0  5026.9     .16       0  5335.9      .1       0
  5380.1     .16       0
Bank Sta=4966,5022.9
XS Rating Curve= 0 ,0
Exp/Cntr=0.3,0.1

Type RM Length L Ch R = 1 ,136594  ,55,55,55
BEGIN DESCRIPTION:
Mapping XS e78118ba
END DESCRIPTION:
XS GIS Cut Line= 3
        2796773.     10095042.03      2796905.38     10094642.72
      2796970.45     10093868.33
#Sta/Elev= 30
  4427.3  1907.4  4478.2 1903.81  4493.2  1903.6  4509.8  1901.5  4532.5    1900
    4583 1897.01  4625.7 1896.22  4683.3 1893.35  4720.5 1889.73  4746.7 1888.74
  4762.6 1887.07  4810.1 1884.53    4867 1882.81  4887.1 1881.08  4917.2 1875.35
  4927.3 1874.67  5024.6 1874.57  5027.4 1874.07  5030.6 1874.57  5063.4 1874.87
  5107.9 1880.92    5128 1881.36    5138 1882.47  5158.1 1888.47  5183.3 1893.12
  5288.5 1904.22  5395.7 1905.92  5489.2 1907.48  5533.1 1909.53  5625.1 1913.04
#Mann= 6 ,-1 , 0
  4427.3      .1       0  4532.5     .16       0  5024.6     .07       0
  5030.6     .16       0  5395.7      .1       0  5533.1     .16       0
Bank Sta=4887.1,5107.9
XS Rating Curve= 0 ,0
Exp/Cntr=0.3,0.1

Type RM Length L Ch R = 1 ,136539  ,56,56,56
BEGIN DESCRIPTION:
Mapping XS 251939a3
END DESCRIPTION:
XS GIS Cut Line= 3
      2796831.58     10095063.76      2796970.48     10094536.38
      2796996.52     10093872.36
#Sta/Elev= 30
  4415.1    1908  4435.8 1907.39  4510.8 1901.71  4577.5 1897.07  4632.3 1895.71
  4652.9 1896.36  4663.3 1893.88    4684  1893.2  4704.7 1890.96  4773.9 1886.19
  4870.1 1881.07  4898.2 1880.34  4904.2 1880.34  4935.1 1880.98  4959.3 1884.22
  4983.1 1884.47  5037.4 1883.31  5053.2 1884.51    5092 1884.33  5113.2 1882.13
  5123.2  1881.9  5133.2 1883.49  5153.3 1888.41  5173.3 1891.84  5290.1 1904.25
  5375.7 1905.39  5493.5 1907.81    5536 1909.54  5583.6 1912.14    5625    1913
#Mann= 8 ,-1 , 0
  4415.1      .1       0  4510.8     .16       0  4898.2     .07       0
  4904.2     .16       0  5053.2      .1       0    5092     .16       0
  5375.7      .1       0    5536     .16       0
#XS Ineff= 2 , 0
       0  4973.1  1884.5  5073.2       0 1884.88
Permanent Ineff=
       T       T
Bank Sta=4983.1,5053.2
XS Rating Curve= 0 ,0
Exp/Cntr=0.3,0.1

Type RM Length L Ch R = 1 ,136483  ,233,233,233
BEGIN DESCRIPTION:
Mapping XS c9c471df
END DESCRIPTION:
XS GIS Cut Line= 3
      2796892.35      10095065.9      2797022.56     10094666.59
       2797048.6     10093848.61
#Sta/Elev= 30
  4413.9 1907.95  4478.8 1903.86  4545.9 1898.75  4584.5 1896.26  4637.1 1894.81
  4692.6  1891.4  4706.6 1890.25  4721.2  1890.6  4738.5 1888.02  4815.9 1882.29
  4856.8 1881.42    4867 1880.04  4903.1 1878.77  4956.8 1874.24  4986.8 1870.28
  5003.8 1870.02  5006.6 1869.52  5009.8 1870.02  5036.9 1874.53  5056.9 1876.49
  5124.5 1885.76  5174.3 1892.04    5287 1903.14    5307 1904.24  5370.4 1905.25
  5437.1 1906.46  5537.3 1909.86  5627.2 1913.11  5647.2 1915.36  5652.3  1916.7
#Mann= 10 ,-1 , 0
  4413.9      .1       0  4478.8     .16       0  4545.9      .1       0
  4692.6     .16       0  4903.1      .1       0  5003.8     .07       0
  5009.8      .1       0  5124.5     .16       0  5370.4      .1       0
  5537.3     .16       0
Bank Sta=4956.8,5036.9
XS Rating Curve= 0 ,0
Exp/Cntr=0.3,0.1

Type RM Length L Ch R = 1 ,136250  ,880,880,880
BEGIN DESCRIPTION:
NORTH GRAPE CREEK 185.0
END DESCRIPTION:
XS GIS Cut Line= 2
      2797045.89     10095084.11      2797471.22      10093990.4
#Sta/Elev= 30
  4471.5 1906.35  4473.3 1906.35  4611.4 1895.96  4658.8 1895.06  4714.9 1891.51
  4747.5 1888.62  4804.5 1882.71  4851.9 1878.93  4922.5    1875    4944 1871.64
  4994.7 1868.09  4997.4 1867.59  5000.7 1868.09  5008.4  1868.3  5020.5 1871.72
  5039.7 1874.98  5069.6 1877.87  5147.9 1880.65  5208.3 1886.21  5238.2 1887.67
  5262.7 1890.81  5376.9 1896.81  5401.4 1899.59  5406.8 1899.24    5426  1901.6
  5430.4 1901.33  5437.6 1902.42  5480.4 1904.14  5643.7  1907.2    5645  1907.2
#Mann= 8 ,-1 , 0
  4471.5      .1       0  4473.3     .16       0  4714.9      .1       0
  4747.5     .16       0  4994.7     .07       0  5000.7     .16       0
  5430.4      .1       0  5643.7     .16       0
Bank Sta=4922.5,5039.7
XS Rating Curve= 0 ,0
Exp/Cntr=0.3,0.1

Type RM Length L Ch R = 1 ,135370  ,725,725,725
BEGIN DESCRIPTION:
NORTH GRAPE CREEK 184.0
END DESCRIPTION:
XS GIS Cut Line= 3
      2797922.61     10095335.88      2798070.18      10094702.2
      2797913.92     10093972.99
#Sta/Elev= 30
  4176.9 1900.71  4240.7 1895.94  4394.7 1890.76  4490.8 1886.67  4544.8 1883.26
  4666.2 1879.15  4751.4 1874.69  4910.1 1868.77  4938.5 1867.08  4948.7 1865.78
  4954.4  1863.9  4995.7 1857.75  4998.5 1857.25  5001.7 1857.75  5010.1 1858.76
  5020.3 1862.15  5030.5 1864.69  5036.9 1864.92  5091.9 1865.99  5132.8 1869.43
  5183.9 1876.42  5240.8 1885.33  5285.1 1889.88  5316.9 1891.23  5378.2 1892.24
  5433.4 1894.68  5470.3 1896.71  5490.7  1899.2  5544.4 1901.82  5573.3 1902.41
#Mann= 6 ,-1 , 0
  4176.9     .16       0  4544.8      .1       0  4995.7     .07       0
  5001.7      .1       0  5036.9     .16       0  5544.4      .1       0
Bank Sta=4954.4,5030.5
XS Rating Curve= 0 ,0
Exp/Cntr=0.3,0.1

Type RM Length L Ch R = 1 ,134645  ,709,709,709
BEGIN DESCRIPTION:
NORTH GRAPE CREEK 183.0
END DESCRIPTION:
XS GIS Cut Line= 3
       2798825.4     10095170.99       2798686.5     10094294.22
      2798356.64     10093964.36
#Sta/Elev= 30
  4363.1    1891  4373.4 1890.65  4394.4 1889.28  4572.9 1878.06  4613.6 1876.57
  4697.2 1873.62  4743.9 1867.33  4765.3 1865.29  4795.7 1867.75  4821.9 1867.74
    4827 1866.32  4884.2 1863.52  4937.4 1854.97  4957.7 1855.58    4967 1854.36
  4967.8 1854.26  4995.2 1848.87  4997.9 1848.37  5001.2 1848.87  5008.3 1849.38
  5028.6 1856.57  5038.7 1858.67  5048.8 1859.12    5206 1858.52  5263.9 1859.64
  5301.2 1862.96  5339.2 1866.09  5483.1 1873.21  5615.5 1878.09  5717.3 1884.24
#Mann= 11 ,-1 , 0
  4363.1     .16       0  4373.4      .1       0  4394.4     .16       0
  4613.6      .1       0  4743.9     .16       0    4967      .1       0
  4995.2     .07       0  5001.2      .1       0  5301.2     .16       0
  5339.2      .1       0  5615.5     .16       0
#XS Ineff= 2 , 0
                          5070.7         1859.51
Permanent Ineff=
       F       F
Bank Sta=4967.8,5028.6
XS Rating Curve= 0 ,0
Exp/Cntr=0.3,0.1

Type RM Length L Ch R = 1 ,133936  ,780,780,780
BEGIN DESCRIPTION:
NORTH GRAPE CREEK 182.0
END DESCRIPTION:
XS GIS Cut Line= 2
       2799493.8     10094363.67      2798755.97     10093660.56
#Sta/Elev= 30
  4441.5 1888.02  4518.4 1886.82  4590.2 1885.66  4649.3 1884.19  4721.2 1881.89
  4756.4 1878.47  4841.3 1873.09  4883.8 1867.97  4897.9 1864.03  4904.8 1863.39
  4912.1 1860.88    4919 1860.39  4933.1 1856.38  4940.4 1853.35  4947.3 1852.43
  4954.5 1850.06  4967.9 1849.11    4994 1845.23  4996.7 1844.73    5000 1845.23
  5011.1 1846.33  5025.3 1849.35  5060.5  1851.6  5131.3 1849.53    5230 1850.52
  5279.7 1851.98  5301.1 1854.75  5329.5 1856.77  5396.9 1858.66  5460.7 1860.19
#Mann= 9 ,-1 , 0
  4441.5      .1       0  4518.4     .16       0  4590.2     .05       0
  4649.3     .16       0  4967.9      .1       0    4994     .07       0
    5000      .1       0    5230     .16       0  5396.9      .1       0
#XS Ineff= 2 , 0
                         5058.22          1851.1
Permanent Ineff=
       F       F
Bank Sta=4967.9,5025.3
XS Rating Curve= 0 ,0
Exp/Cntr=0.3,0.1

Type RM Length L Ch R = 1 ,133156  ,763,763,763
BEGIN DESCRIPTION:
NORTH GRAPE CREEK 181.0
END DESCRIPTION:
XS GIS Cut Line= 2
      2799927.78     10093591.07      2798652.61     10093061.92
#Sta/Elev= 30
  4092.6 1890.18  4156.8 1886.06  4265.1 1882.68    4342 1878.45  4435.4 1871.53
  4488.6 1869.79  4547.1 1862.07  4565.6 1860.86  4589.5 1858.42    4648  1847.5
  4685.2    1846  4784.8 1843.65  4895.2 1844.57  4968.8 1842.32  4990.8 1838.16
  4998.3  1838.1  5001.1  1837.6  5004.3  1838.1  5014.7 1838.73    5023 1842.55
  5038.6 1847.74    5121 1848.89  5168.8 1851.16  5209.4 1855.03  5221.9 1855.61
    5297 1871.23  5352.1 1879.33  5412.7 1885.11  5463.9 1887.42  5473.2 1887.78
#Mann= 10 ,-1 , 0
  4092.6      .1       0    4342     .05       0  4565.6      .1       0
  4685.2     .05       0  4895.2      .1       0  4998.3     .07       0
  5004.3      .1       0  5209.4     .16       0    5297      .1       0
  5463.9     .16       0
Bank Sta=4968.8,5023
XS Rating Curve= 0 ,0
Exp/Cntr=0.3,0.1

Type RM Length L Ch R = 1 ,132393  ,1002,1002,1002
BEGIN DESCRIPTION:
NORTH GRAPE CREEK 180.0
END DESCRIPTION:
XS GIS Cut Line= 2
      2800266.35     10092818.52      2799163.91     10092705.67
#Sta/Elev= 30
  4327.4 1864.03  4395.6 1859.07  4415.7 1856.96  4445.9 1852.43    4466 1852.04
  4506.2 1847.25  4521.5 1846.68  4526.5 1845.49  4620.9 1843.47  4890.3 1842.04
  4958.6 1840.93  4968.6 1839.73  4982.3 1835.13  4995.8 1832.09  4998.5 1831.59
  5001.8 1832.09  5013.3 1832.49  5028.9 1835.66    5049 1837.44  5107.6  1838.2
  5169.7 1837.89  5280.2 1841.16  5311.4 1844.85  5320.4 1848.36  5330.5 1850.15
  5340.5 1849.64  5360.7 1852.31    5388 1859.14  5430.8 1866.95  5435.6 1866.95
#Mann= 6 ,-1 , 0
  4327.4     .05       0  4890.3      .1       0  4982.3     .16       0
  4995.8     .07       0  5001.8     .16       0    5388      .1       0
Bank Sta=4968.6,5049
XS Rating Curve= 0 ,0
Exp/Cntr=0.3,0.1

Type RM Length L Ch R = 1 ,131391  ,1381,1381,1381
BEGIN DESCRIPTION:
NORTH GRAPE CREEK 179.0
END DESCRIPTION:
XS GIS Cut Line= 2
       2800552.8     10092566.77      2799606.64     10091794.21
#Sta/Elev= 30
  4303.1 1852.45  4379.4 1844.54  4464.1 1839.12  4585.4 1835.85  4806.1 1834.39
  4884.1 1833.65    4948 1831.51  4976.7 1828.54  4994.5 1824.62  4997.3 1824.12
  5000.5 1824.62  5011.9  1825.1  5040.6 1829.83  5047.1 1829.09    5055  1831.5
  5083.3 1834.71  5168.4 1836.42  5217.9 1838.55  5238.8 1838.01  5246.7 1839.56
  5267.5 1848.78  5275.4 1850.14  5296.2 1851.24  5310.6 1854.73  5324.9 1856.31
  5361.7 1857.26  5388.8 1858.16  5409.6    1857  5438.4 1857.16  5524.6  1852.9
#Mann= 5 ,-1 , 0
  4303.1     .05       0  4806.1      .1       0  4994.5     .07       0
  5000.5      .1       0  5361.7     .05       0
Bank Sta=4948,5055
XS Rating Curve= 0 ,0
Exp/Cntr=0.3,0.1

Type RM Length L Ch R = 1 ,130010  ,803,803,803
BEGIN DESCRIPTION:
NORTH GRAPE CREEK 178.0
END DESCRIPTION:
XS GIS Cut Line= 2
      2801472.96     10092028.59      2800396.58     10090969.57
#Sta/Elev= 30
  4095.4 1852.08  4102.1 1852.08  4123.2  1844.5  4158.5  1845.6  4177.5 1844.47
  4298.3 1837.87  4320.2 1837.75  4377.8 1834.63  4434.4 1834.12  4476.8 1831.16
  4519.2 1831.64  4591.5 1829.39  4738.2 1825.55  4884.8 1823.58  4929.4 1824.04
  4964.7 1820.62    4997 1809.39  4999.8 1808.89    5003 1809.39  5035.4 1821.76
  5037.2 1822.25  5056.6  1825.2    5099 1824.01    5198 1826.28    5342 1836.15
  5424.3 1844.25  5466.7 1853.17    5530 1861.17  5558.7 1866.12  5605.4 1868.85
#Mann= 12 ,-1 , 0
  4095.4     .05       0  4177.5      .1       0  4298.3     .05       0
  4320.2      .1       0  4591.5     .05       0  4738.2      .1       0
  4884.8     .16       0    4997     .07       0    5003     .16       0
  5037.2     .05       0    5342      .1       0    5530     .05       0
Bank Sta=4964.7,5035.4
XS Rating Curve= 0 ,0
Exp/Cntr=0.3,0.1

Type RM Length L Ch R = 1 ,129207  ,749,749,749
BEGIN DESCRIPTION:
NORTH GRAPE CREEK 177.0
END DESCRIPTION:
XS GIS Cut Line= 2
      2802167.41     10091481.72      2800909.51     10090458.05
#Sta/Elev= 30
    3942 1854.29  3993.1  1849.6  4039.6 1846.71  4060.4 1843.78  4095.6 1844.66
  4173.9 1839.78  4231.3 1838.52  4266.5 1835.54    4324 1834.73    4380 1831.18
  4437.4 1830.86  4506.2 1827.31  4544.5  1827.2  4643.6 1821.57  4781.4 1817.41
  4869.9 1815.97  4907.2 1817.37  4942.3 1816.19  4995.3 1805.98  4998.1 1805.48
  5001.3 1805.98    5013 1810.85  5020.6 1814.74  5027.1 1817.75    5035 1818.44
  5154.9 1816.86  5247.6 1817.84  5406.3 1824.84    5532 1835.01  5563.8 1840.49
#Mann= 9 ,-1 , 0
    3942      .1       0  3993.1     .05       0  4506.2      .1       0
  4781.4     .05       0  4869.9      .1       0  4995.3     .07       0
  5001.3      .1       0    5013     .05       0  5406.3      .1       0
#XS Ineff= 2 , 0
                         5039.64          1818.4
Permanent Ineff=
       F       F
Bank Sta=4942.3,5020.6
XS Rating Curve= 0 ,0
Exp/Cntr=0.3,0.1

Type RM Length L Ch R = 1 ,128458  ,666,666,666
BEGIN DESCRIPTION:
NORTH GRAPE CREEK 176.0
END DESCRIPTION:
XS GIS Cut Line= 2
      2802618.78     10090960.87      2801203.85     10089815.04
#Sta/Elev= 30
  4093.1  1852.4    4097 1851.86  4219.7  1842.7  4234.1 1840.68  4247.9 1841.01
  4309.1 1837.14  4368.4 1834.48  4427.1 1830.15  4432.4 1830.09    4525 1825.19
  4638.6  1821.1  4937.5 1812.86  4953.3 1810.37  4980.6 1803.65  4998.4 1798.54
  5001.2 1798.04  5004.4 1798.54  5030.2 1803.45  5034.2 1803.62    5051 1804.98
  5065.4 1808.83  5072.2 1808.86  5178.9 1808.52  5442.7 1813.49  5498.7  1813.5
  5626.6 1818.72  5690.5 1819.65  5727.2 1822.26  5861.6 1827.17  5913.8 1830.26
#Mann= 11 ,-1 , 0
  4093.1     .16       0    4097     .05       0  4309.1      .1       0
  4427.1     .05       0  4432.4      .1       0  4953.3     .05       0
  4998.4    .035       0  5004.4     .05       0  5034.2      .1       0
  5072.2     .05       0  5861.6      .1       0
Bank Sta=4980.6,5030.2
XS Rating Curve= 0 ,0
Exp/Cntr=0.3,0.1

Type RM Length L Ch R = 1 ,127792  ,980,980,980
BEGIN DESCRIPTION:
Mapping XS e4e6dbec
END DESCRIPTION:
XS GIS Cut Line= 2
      2802922.62      10090283.8      2801491.86     10089347.31
#Sta/Elev= 30
  4223.5 1835.77    4306 1831.22    4336 1827.51  4378.3 1825.97  4414.5 1821.74
  4456.7 1820.61  4486.9 1817.51  4538.2 1815.81  4580.4 1812.37  4754.3 1806.38
  4812.6 1806.11  4890.9  1803.7  4934.4 1804.19  4942.2 1803.91  4963.3 1799.28
  4996.5  1791.9  4999.3  1791.4  5002.5  1791.9  5020.6 1792.81  5035.7 1796.22
  5056.8 1798.62  5071.9 1802.38  5085.4 1802.91  5237.7 1803.94  5433.7 1807.36
  5744.3 1822.52  5768.9 1824.63  5775.2 1825.03  5858.9 1828.49  5933.5 1834.81
#Mann= 7 ,-1 , 0
  4223.5     .05       0  4934.4      .1       0  4996.5     .07       0
  5002.5      .1       0  5085.4     .05       0  5768.9      .1       0
  5775.2     .05       0
Bank Sta=4963.3,5056.8
XS Rating Curve= 0 ,0
Exp/Cntr=0.3,0.1

Type RM Length L Ch R = 1 ,126812  ,913,913,913
BEGIN DESCRIPTION:
Mapping XS d574cd0b
END DESCRIPTION:
XS GIS Cut Line= 2
      2803591.01     10089754.28      2802002.98     10088712.95
#Sta/Elev= 30
  4300.3 1837.19  4352.8 1833.98  4397.3 1831.46  4418.4 1828.47  4433.5 1828.79
  4460.5 1826.18  4482.7  1826.1  4605.2 1817.65  4635.4 1817.41  4662.5 1814.88
  4816.3 1808.23  4924.8 1801.55    4961 1798.78    4973 1796.45  4982.1 1791.69
  4993.9 1784.98  4996.7 1784.48  4999.9 1784.98  5029.2 1787.19  5054.4 1790.34
  5068.7 1791.89  5161.9 1794.86  5336.9 1798.37  5594.8 1798.01  5785.3 1800.28
  5856.2 1802.34  5942.7 1807.05  6064.1 1816.94  6085.2  1817.2  6199.3 1829.48
#Mann= 9 ,-1 , 0
  4300.3     .05       0  4352.8      .1       0  4993.9     .07       0
  4999.9      .1       0  5029.2     .05       0  5161.9      .1       0
  5336.9     .05       0  5785.3      .1       0  5942.7     .05       0
Bank Sta=4982.1,5054.4
XS Rating Curve= 0 ,0
Exp/Cntr=0.3,0.1

Type RM Length L Ch R = 1 ,125899  ,532,532,532
BEGIN DESCRIPTION:
Mapping XS 9865f2cb
END DESCRIPTION:
XS GIS Cut Line= 4
      2804155.26     10089815.08      2803894.83      10089033.8
      2803252.47     10088417.48       2802280.3      10088278.6
#Sta/Elev= 30
    3755 1838.89  3788.9 1837.09    3914 1830.44  3925.1 1830.54    3948 1836.86
  3977.3 1832.89  3982.5 1834.29  3988.3  1830.4  4008.9  1827.2  4193.5 1820.62
  4372.9  1814.5  4493.8 1808.89  4519.9 1807.99  4796.3 1797.82  4915.6  1790.2
    4958 1782.67  4990.2 1776.68    4993 1776.18  4996.2 1776.68  5033.7 1780.39
    5064 1782.31  5083.6 1782.31    5215 1785.09  5302.6 1786.53  5346.3 1786.55
  5800.2  1790.5  5876.5 1792.21  5980.2 1794.66  6139.5 1800.69  6450.8 1819.75
#Mann= 18 ,-1 , 0
    3755      .1       0  3788.9     .05       0    3948      .1       0
  4193.5     .05       0  4372.9      .1       0  4493.8     .05       0
  4519.9      .1       0  4796.3     .16       0  4990.2     .07       0
  4996.2     .16       0  5033.7     .05       0  5083.6      .1       0
    5215     .05       0  5302.6      .1       0  5346.3     .05       0
  5800.2      .1       0  5876.5     .05       0  5980.2      .1       0
Bank Sta=4958,5064
XS Rating Curve= 0 ,0
Exp/Cntr=0.3,0.1

Type RM Length L Ch R = 1 ,125367  ,746,746,746
BEGIN DESCRIPTION:
NORTH GRAPE CREEK 175.0
END DESCRIPTION:
XS GIS Cut Line= 2
      2804085.76     10088348.03      2802723.25     10088052.96
#Sta/Elev= 30
  4552.5 1789.99  4580.4 1791.61  4621.4 1792.17  4674.9 1791.33  4694.5 1791.79
  4794.5 1785.09  4880.4 1783.74  4948.8 1782.28  4969.2 1780.01  4974.4 1777.77
  4979.5 1776.91  4989.7 1771.31  4996.9 1769.05  4999.7 1768.55  5002.9 1769.05
  5018.5 1772.71  5023.6 1772.44  5030.6  1775.2  5051.1 1777.59  5072.8 1781.53
  5166.1 1782.03  5300.8  1785.3  5526.9 1787.88    5665 1790.36  5730.9 1793.68
  5749.8 1793.41  5818.5 1795.31  5873.4 1798.31  5917.5 1798.72  5946.6 1800.69
#Mann= 9 ,-1 , 0
  4552.5     .05       0  4674.9      .1       0  4794.5     .05       0
  4880.4      .1       0  4996.9     .07       0  5002.9      .1       0
  5300.8     .05       0  5526.9      .1       0  5749.8     .05       0
Bank Sta=4979.5,5030.6
XS Rating Curve= 0 ,0
Exp/Cntr=0.3,0.1

Type RM Length L Ch R = 1 ,124621  ,651,651,651
BEGIN DESCRIPTION:
NORTH GRAPE CREEK 174.0
END DESCRIPTION:
XS GIS Cut Line= 4
      2804389.64     10088295.98      2804120.53     10087723.04
      2803851.43      10087558.1      2802705.57     10087818.53
#Sta/Elev= 30
  4269.4 1784.73  4371.3 1783.18  4415.5 1780.92  4616.6 1775.97    4847 1774.57
  4947.4 1772.67  4968.7 1766.16  4995.6 1761.98  4998.4 1761.48  5001.6 1761.98
  5020.8 1764.37  5063.4 1773.25  5151.1 1770.35  5295.7 1772.89  5357.9 1775.17
  5395.4 1775.02  5449.1 1777.55    5621 1779.73  5712.7 1781.97  5733.8 1783.53
  5918.4 1786.15  6008.3  1789.8  6072.2 1791.16  6113.3 1793.38    6185 1794.79
  6236.3 1797.33  6297.8 1797.68  6351.6 1800.38  6381.4 1800.34  6393.1 1800.39
#Mann= 8 ,-1 , 0
  4269.4      .1       0    4847     .16       0  4995.6     .07       0
  5001.6     .16       0  5295.7      .1       0  6008.3     .05       0
  6113.3      .1       0  6381.4     .05       0
Bank Sta=4947.4,5063.4
XS Rating Curve= 0 ,0
Exp/Cntr=0.3,0.1

Type RM Length L Ch R = 1 ,123970  ,888,888,888
BEGIN DESCRIPTION:
NORTH GRAPE CREEK 172.0
END DESCRIPTION:
XS GIS Cut Line= 2
      2804910.44     10087610.17      2803729.94     10086559.87
#Sta/Elev= 30
  4237.8  1772.1    4263 1772.34  4300.4 1771.44  4541.2 1770.94  4654.9 1773.14
  4767.1 1772.18  4824.7 1772.27  4859.8 1773.59  4909.7 1769.74  4930.9 1766.31
  4951.8 1765.45  4987.7 1758.27    4999 1757.02  5001.7 1756.52    5005 1757.02
  5029.6 1761.21  5051.3 1764.15  5078.1 1766.61  5114.8 1771.59  5185.9 1776.45
  5222.1 1780.83  5277.9 1785.82  5320.5 1791.04  5377.4 1802.81  5469.4 1808.97
  5582.7 1814.79  5628.8 1818.16  5693.9 1823.17  5773.8 1830.27  5817.9 1832.92
#Mann= 11 ,-1 , 0
  4237.8     .05       0    4263      .1       0  4767.1     .16       0
    4999     .07       0    5005     .16       0  5029.6      .1       0
  5078.1     .16       0  5222.1      .1       0  5582.7     .16       0
  5628.8     .05       0  5693.9      .1       0
#XS Ineff= 2 , 0
         4860.87 1773.59
Permanent Ineff=
       F       F
Bank Sta=4951.8,5051.3
XS Rating Curve= 0 ,0
Exp/Cntr=0.3,0.1

Type RM Length L Ch R = 1 ,123082  ,742,742,742
BEGIN DESCRIPTION:
NORTH GRAPE CREEK 170.0
END DESCRIPTION:
XS GIS Cut Line= 2
      2804945.18     10087540.74      2805136.16     10085952.18
#Sta/Elev= 30
  4158.2 1771.33  4377.5 1768.35  4578.2  1767.6  4650.1 1765.31  4678.9 1763.46
  4699.1 1760.91  4739.4 1759.01  4779.6 1758.54  4840.1 1759.65  4901.7 1758.87
  4920.7    1760  4950.9  1759.2    4971 1757.01  4988.2 1752.41  4990.9 1751.91
  4994.2 1752.41  5021.4 1754.67  5041.5 1759.03    5102 1763.93  5122.1 1767.56
  5148.2 1769.79  5231.4  1772.6  5235.5 1772.17  5414.2 1781.41  5496.2 1783.61
  5564.2 1784.72  5605.6 1788.47  5656.4 1796.33  5726.4 1798.45  5758.2 1801.06
#Mann= 6 ,-1 , 0
  4158.2     .05       0  4377.5      .1       0  4988.2     .07       0
  4994.2      .1       0  5231.4     .05       0  5496.2      .1       0
Bank Sta=4950.9,5041.5
XS Rating Curve= 0 ,0
Exp/Cntr=0.3,0.1

Type RM Length L Ch R = 1 ,122340  ,949,949,949
BEGIN DESCRIPTION:
NORTH GRAPE CREEK 167.0
END DESCRIPTION:
XS GIS Cut Line= 2
      2805136.13      10087662.3       2805864.4     10086751.97
#Sta/Elev= 30
  4342.7 1775.09  4470.9 1773.46    4671 1766.21    4948  1762.9  4955.6 1762.33
  4968.8 1757.53  4976.8  1752.4  4994.6 1747.22  4997.3 1746.72  5000.6 1747.22
    5012 1748.42  5026.4 1753.44  5055.2 1756.56  5090.4 1755.08  5119.2 1757.86
    5140 1759.18  5160.9  1757.9  5175.3 1760.29  5189.7 1766.61  5218.5 1787.11
  5232.9 1794.47  5296.9 1814.55  5303.3 1818.22    5361 1831.47  5396.2 1843.03
  5410.6 1844.53  5445.8 1854.86  5474.6 1857.54    5481 1860.23  5508.5  1863.1
#Mann= 4 ,-1 , 0
  4342.7     .05       0  4994.6     .04       0  5000.6     .05       0
  5119.2     .16       0
#XS Ineff= 2 , 0
                         5141.78         1759.13
Permanent Ineff=
       F       F
Bank Sta=4968.8,5026.4
XS Rating Curve= 0 ,0
Exp/Cntr=0.3,0.1

Type RM Length L Ch R = 1 ,121391  ,1074,1074,1074
BEGIN DESCRIPTION:
NORTH GRAPE CREEK 166.0
END DESCRIPTION:
XS GIS Cut Line= 2
      2805222.96      10088096.3      2806732.46      10087428.3
#Sta/Elev= 30
  3867.3 1773.25  3939.9 1773.27  4235.8 1766.95  4387.3 1760.93  4516.9  1759.4
  4759.1  1756.2    4781 1753.46  4820.6 1754.58  4835.6 1752.01  4897.5 1749.03
  4966.9 1748.89  4979.2 1744.84  4993.1 1739.76  4995.9 1739.26  4999.1 1739.76
  5010.6 1740.98  5032.5 1750.58  5048.2 1756.22  5071.4 1772.32  5094.7 1780.17
  5100.2  1779.2  5123.5 1783.57  5170.1 1798.11  5216.7 1806.41  5251.2 1817.95
  5338.6 1836.82  5396.1 1851.89  5448.1 1859.07  5515.5 1861.08    5518 1861.33
#Mann= 7 ,-1 , 0
  3867.3      .1       0  4516.9     .05       0  4820.6      .1       0
  4979.2     .16       0  4993.1     .07       0  4999.1     .16       0
  5515.5      .1       0
Bank Sta=4966.9,5032.5
XS Rating Curve= 0 ,0
Exp/Cntr=0.3,0.1

Type RM Length L Ch R = 1 ,120317  ,814,814,814
BEGIN DESCRIPTION:
NORTH GRAPE CREEK 164.0
END DESCRIPTION:
XS GIS Cut Line= 3
      2805361.89     10089320.23      2806846.22     10088521.65
      2807089.27     10087879.31
#Sta/Elev= 30
  3581.8 1787.71  3600.4 1787.03  3688.1 1783.69    3792 1782.29  3800.7 1783.33
  3829.8 1781.81  3944.6 1775.46  4153.1 1764.93  4306.5 1765.99  4350.3 1759.78
  4377.2 1758.97  4518.2  1753.6  4656.2 1746.64  4683.8 1746.95    4700 1745.14
  4714.9 1745.95  4935.3 1739.78  4963.3 1741.04  4998.1 1737.51  5000.8 1737.01
  5004.1 1737.51  5031.4 1741.63  5102.7 1741.18  5265.8 1750.18  5446.9  1754.3
  5615.8 1760.06  5719.3 1765.94  5825.5 1773.31  5880.5 1781.78  5954.1 1785.67
#Mann= 14 ,-1 , 0
  3581.8     .05       0  3600.4      .1       0  3800.7     .05       0
  3829.8      .1       0  3944.6     .05       0  4377.2     .16       0
  4518.2     .05       0  4714.9      .1       0  4998.1     .07       0
  5004.1      .1       0  5102.7     .16       0  5446.9      .1       0
  5615.8     .05       0  5719.3      .1       0
#XS Ineff= 2 , 0
         4711.95    1746
Permanent Ineff=
       F       F
Bank Sta=4963.3,5031.4
XS Rating Curve= 0 ,0
Exp/Cntr=0.3,0.1

Type RM Length L Ch R = 1 ,119503  ,597,597,597
BEGIN DESCRIPTION:
NORTH GRAPE CREEK 163.0
END DESCRIPTION:
XS GIS Cut Line= 3
      2806281.98     10090752.56      2806646.57     10089476.51
      2807201.57     10088748.06
#Sta/Elev= 30
  3482.7 1798.22  3494.6 1797.71  3694.2 1791.48  4147.8 1774.96  4422.5 1768.07
  4523.5 1765.08  4624.5 1761.63  4646.3 1762.12  4677.5 1758.47  4730.2 1740.12
  4739.9 1738.32  4758.8 1736.75  4797.8  1736.4  4814.7 1733.82  4817.4 1730.75
  4820.1 1730.25  4823.4 1730.75  4863.6 1734.41  4899.4 1735.41    4941 1734.28
  4949.3 1735.24  4970.1 1731.41  4984.6 1733.19  4990.9 1731.79  5001.6 1732.15
  5034.5 1736.44  5090.7 1739.83  5231.7 1744.23  5594.8 1748.01  5725.6 1749.45
#Mann= 11 ,-1 , 0
  3482.7      .1       0  3494.6     .05       0  3694.2      .1       0
  4422.5     .05       0  4523.5      .1       0  4624.5     .05       0
  4817.4     .04       0  4823.4     .05       0  5001.6      .1       0
  5231.7     .16       0  5594.8      .1       0
Bank Sta=4797.8,5034.5
XS Rating Curve= 0 ,0
Exp/Cntr=0.3,0.1

Type RM Length L Ch R = 1 ,118906  ,638,638,638
BEGIN DESCRIPTION:
NORTH GRAPE CREEK 161.0
END DESCRIPTION:
XS GIS Cut Line= 3
      2806959.07     10090518.19      2807176.08     10089424.42
      2807462.54     10088790.75
#Sta/Elev= 30
  4261.3 1779.98  4316.8 1779.36  4357.6 1776.72  4408.6 1776.28  4500.3 1771.88
  4622.7 1769.02  4632.9 1768.09  4645.9 1764.85  4720.8 1762.03  4775.6  1759.3
  4820.2 1754.38  4877.5 1749.13  4896.7  1746.7  4901.8 1744.74  4935.6 1740.93
  4969.3 1733.85  4989.7 1724.53  5001.1  1723.1  5003.9  1722.6  5007.1  1723.1
  5010.1 1725.51  5030.5 1729.94  5152.6 1733.12  5208.8 1732.55  5251.9 1737.98
  5355.1 1740.11  5511.6 1740.24  5714.4 1739.97  5885.9 1744.93  6071.8 1748.94
#Mann= 11 ,-1 , 0
  4261.3     .05       0  4720.8      .1       0  4820.2     .16       0
  4935.6      .1       0  5001.1     .07       0  5007.1      .1       0
  5251.9     .05       0  5355.1      .1       0  5511.6     .16       0
  5714.4      .1       0  5885.9     .05       0
#XS Ineff= 2 , 0
                         5398.31         1740.49
Permanent Ineff=
       F       F
Bank Sta=4969.3,5030.5
XS Rating Curve= 0 ,0
Exp/Cntr=0.3,0.1

Type RM Length L Ch R = 1 ,118268  ,376,376,376
BEGIN DESCRIPTION:
Mapping XS 2defe4ad
END DESCRIPTION:
XS GIS Cut Line= 2
      2807662.01     10090045.84      2807722.77     10089334.03
#Sta/Elev= 30
  4562.7 1742.37  4594.9  1741.7  4702.9 1740.82  4755.5 1740.48  4797.6 1739.58
  4875.9 1736.15  4906.1 1733.38  4916.1 1731.64  4931.9 1726.92  4946.2 1726.06
  4966.3  1725.7  4976.3 1724.23  4993.4 1718.87  4996.1 1718.37  4999.4 1718.87
  5006.4 1719.18  5012.8 1721.51  5026.5 1726.62  5050.9 1726.73  5066.6 1726.28
  5086.7 1725.05  5096.7 1725.73  5111.8 1730.85  5116.8 1732.31  5136.9 1734.48
    5157 1735.11  5169.9 1736.04    5177 1736.03  5197.1 1737.43  5277.1 1739.54
#Mann= 7 ,-1 , 0
  4562.7      .1       0  4702.9     .05       0  4797.6      .1       0
  4993.4     .07       0  4999.4      .1       0  5012.8     .05       0
  5111.8      .1       0
Bank Sta=4966.3,5026.5
XS Rating Curve= 0 ,0
Exp/Cntr=0.3,0.1

Type RM Length L Ch R = 1 ,117892  ,430,430,430
BEGIN DESCRIPTION:
NORTH GRAPE CREEK 159.0
END DESCRIPTION:
XS GIS Cut Line= 3
      2807939.79     10090149.97      2808347.77     10088474.64
      2808252.87     10088284.84
#Sta/Elev= 30
  4492.7 1736.41  4707.1 1737.13  4859.4 1735.92  4909.1 1731.15  4933.7 1729.06
    4952 1724.79  5000.4 1716.22  5003.2 1715.72  5006.4 1716.22  5053.7 1725.08
  5100.6 1722.53  5116.7 1727.94  5133.7 1730.62  5238.7 1734.73  5342.6 1730.46
    5374 1732.18  5392.6 1737.62  5397.7 1736.15  5434.3 1739.84  5439.1 1738.02
  5517.7 1734.71  5564.6 1738.63  5753.2 1747.12  5849.7 1754.43  5945.2 1763.14
  6055.6 1769.29  6247.5 1783.17  6320.1 1786.46  6359.3 1792.03  6429.2 1793.61
#Mann= 13 ,-1 , 0
  4492.7      .1       0  4707.1     .05       0  4909.1     .16       0
  5000.4     .07       0  5006.4     .16       0  5133.7     .05       0
  5238.7      .1       0  5342.6     .16       0  5439.1      .1       0
  5753.2     .16       0  5849.7      .1       0  5945.2     .16       0
  6055.6      .1       0
#XS Ineff= 2 , 0
                         5225.79         1734.71
Permanent Ineff=
       F       F
Bank Sta=4952,5053.7
XS Rating Curve= 0 ,0
Exp/Cntr=0.3,0.1

Type RM Length L Ch R = 1 ,117462  ,776,776,776
BEGIN DESCRIPTION:
NORTH GRAPE CREEK 158.0
END DESCRIPTION:
XS GIS Cut Line= 2
      2808339.08     10090106.62      2808790.47     10088544.11
#Sta/Elev= 30
  4507.7 1729.89  4625.2 1730.15    4693 1731.91  4760.5 1733.17  4814.8 1732.12
  4833.4 1730.47  4848.4 1726.78  4854.2 1723.14  4864.6 1720.33  4979.1 1719.09
  4996.9 1713.67  4999.7 1713.17  5002.9 1713.67  5020.7 1718.08  5026.9 1722.37
  5058.2 1723.22  5083.2 1720.15  5198.5 1727.07  5429.2 1734.51  5541.2 1738.84
  5602.9 1743.74  5634.9 1748.32  5655.7  1755.1  5712.7 1762.79  5759.8 1773.73
  5805.1 1780.31  5832.6 1787.59  5863.9 1791.74  6036.2 1796.04  6134.1 1800.43
#Mann= 9 ,-1 , 0
  4507.7      .1       0    4693     .16       0  4996.9     .07       0
  5002.9     .16       0  5058.2     .05       0  5198.5     .16       0
  5429.2      .1       0  5602.9     .16       0  5805.1      .1       0
Bank Sta=4979.1,5026.9
XS Rating Curve= 0 ,0
Exp/Cntr=0.3,0.1

Type RM Length L Ch R = 1 ,116686  ,570,570,570
BEGIN DESCRIPTION:
NORTH GRAPE CREEK 157.0
END DESCRIPTION:
XS GIS Cut Line= 4
      2808564.98     10090144.91      2809181.29     10089867.13
       2809354.9     10089537.27      2809155.25     10088599.78
#Sta/Elev= 30
    4210 1727.34  4611.3 1723.15  4833.5  1718.2  4856.6  1718.4  4879.8 1716.88
  4884.1 1714.91  4901.2 1713.06    4969 1715.72  5000.3 1709.49    5003 1708.99
  5006.3 1709.49    5014 1712.41  5048.1 1712.86  5063.7 1715.35  5070.7 1718.14
  5071.7  1718.4  5080.1 1720.59  5115.9 1724.55  5212.5 1728.71  5319.5 1733.01
  5414.5 1737.64  5509.3 1744.35  5647.8 1758.59  5722.5 1763.25  5753.2 1766.56
  5783.8 1767.72  5855.4 1777.02  5978.1 1788.38  6182.8 1801.19  6217.3 1801.66
#Mann= 8 ,-1 , 0
    4210     .05       0  4611.3      .1       0  5000.3     .07       0
  5006.3      .1       0  5071.7     .16       0  5212.5      .1       0
  5319.5     .05       0  5414.5      .1       0
Bank Sta=4969,5070.7
XS Rating Curve= 0 ,0
Exp/Cntr=0.3,0.1

Type RM Length L Ch R = 1 ,116116  ,458,458,458
BEGIN DESCRIPTION:
NORTH GRAPE CREEK 155.0
END DESCRIPTION:
XS GIS Cut Line= 3
       2809493.6     10091261.12      2809849.51     10089568.39
      2809502.87     10088684.47
#Sta/Elev= 30
  3530.7 1741.41  3770.6 1732.74  4090.1 1725.44  4164.3 1721.42    4209 1710.91
  4222.9 1709.38  4253.6 1712.17  4339.3 1712.88  4402.5 1713.31  4433.7 1713.74
  4580.5    1715  4832.1 1712.23  4891.5 1708.96  4968.9  1711.3  4996.5 1706.04
  4999.3 1705.54  5002.5 1706.04    5036 1710.85  5257.3 1724.48  5335.5 1726.93
  5442.9 1731.21  5574.9  1737.5  5688.8 1745.62  5730.2 1755.19  5759.5  1759.1
  5899.2 1765.61  6019.6 1778.07  6128.1 1783.43  6182.4  1783.1  6209.9 1787.48
#Mann= 12 ,-1 , 0
  3530.7      .1       0  4339.3     .05       0  4402.5      .1       0
  4433.7     .05       0  4832.1     .16       0  4996.5     .07       0
  5002.5     .16       0  5257.3      .1       0  5335.5     .16       0
  5442.9     .05       0  5574.9     .16       0  5730.2      .1       0
Bank Sta=4968.9,5036
XS Rating Curve= 0 ,0
Exp/Cntr=0.3,0.1

Type RM Length L Ch R = 1 ,115658  ,829,829,829
BEGIN DESCRIPTION:
NORTH GRAPE CREEK 154.0
END DESCRIPTION:
XS GIS Cut Line= 3
      2810127.29     10091382.61      2810240.13     10089351.37
      2809745.34      10088578.8
#Sta/Elev= 30
  3524.1 1745.64  3567.6 1743.77  3963.7  1722.6  4116.2 1718.59  4418.2 1713.38
  4524.5 1705.64  4562.3 1708.22  4570.6 1708.17  4644.7 1709.84  4866.5 1708.29
  4869.1 1708.26  4975.2 1707.78  4985.2 1706.44  4992.2 1702.32    4995 1701.82
  4998.2 1702.32  5000.4 1702.43  5025.3  1707.4  5215.6  1718.5  5310.9 1721.84
  5526.1 1728.13  5703.6 1736.19  5748.6 1739.18  5840.7 1743.74  5884.1 1751.42
  5935.6 1754.26  6077.3 1759.52  6121.4 1761.51  6181.1 1763.58  6475.9 1772.28
#Mann= 18 ,-1 , 0
  3524.1     .16       0  3567.6      .1       0  4116.2     .05       0
  4418.2      .1       0  4562.3     .16       0  4570.6      .1       0
  4866.5     .05       0  4869.1      .1       0  4992.2     .07       0
  4998.2      .1       0  5000.4     .16       0  5310.9      .1       0
  5703.6     .05       0  5748.6      .1       0  5935.6     .16       0
  6077.3      .1       0  6121.4     .16       0  6181.1      .1       0
Bank Sta=4975.2,5025.3
XS Rating Curve= 0 ,0
Exp/Cntr=0.3,0.1

Type RM Length L Ch R = 1 ,114829  ,523,523,523
BEGIN DESCRIPTION:
NORTH GRAPE CREEK 153.0
END DESCRIPTION:
XS GIS Cut Line= 3
      2810596.04     10091382.62      2811151.59     10089507.62
      2811671.23     10088927.36
#Sta/Elev= 30
  3727.7  1733.2  4034.8 1724.46  4068.1 1721.52  4101.3 1721.06    4187 1716.15
  4316.4 1710.73  4498.3 1706.28  4905.1 1702.93  4967.7  1704.1  4982.4  1701.3
  4989.8 1697.88    4996  1697.7  4998.7  1697.2    5002  1697.7  5082.4 1703.97
  5127.4 1706.08  5194.5 1705.71  5238.9 1703.18  5266.2 1705.84  5332.7 1705.63
  5431.2 1708.35  5443.9 1708.66  5635.2 1714.33  5747.2  1714.4  5748.2  1714.4
  6129.2 1719.79  6166.7 1720.83  6250.6 1722.01  6314.2 1725.09  6462.2 1728.45
#Mann= 12 ,-1 , 0
  3727.7     .16       0    4187      .1       0  4982.4     .05       0
    4996     .04       0    5002     .05       0  5127.4     .16       0
  5431.2      .1       0  5443.9     .16       0  5747.2     .05       0
  5748.2      .1       0  6129.2     .05       0  6166.7      .1       0
#XS Ineff= 2 , 0
                         5144.27         1706.27
Permanent Ineff=
       F       F
Bank Sta=4967.7,5082.4
XS Rating Curve= 0 ,0
Exp/Cntr=0.3,0.1

Type RM Length L Ch R = 1 ,114306  ,838,838,838
BEGIN DESCRIPTION:
NORTH GRAPE CREEK 151.0
END DESCRIPTION:
XS GIS Cut Line= 4
      2810899.84     10091339.24      2811333.88     10090636.09
      2811767.91     10089368.73      2812314.16      10089082.6
#Sta/Elev= 30
  3917.6 1727.21  3945.4 1726.71  4073.9 1723.16  4131.8 1717.63    4211 1716.69
    4269 1713.18  4311.9 1705.63  4387.3 1703.01  4947.3 1702.69  4997.1  1694.9
  4999.9  1694.4  5003.1  1694.9  5049.5 1702.17  5066.1 1702.67  5190.4 1702.19
  5205.9 1701.24  5211.5 1697.79  5243.2 1701.78  5303.3 1701.88  5370.1 1700.35
  5412.3 1706.01  6002.8  1720.4  6146.2 1724.89  6323.7 1735.83  6355.1 1739.66
  6384.3 1749.54  6485.8 1757.69  6544.1 1763.53  6637.6 1767.53  6700.2 1768.32
#Mann= 12 ,-1 , 0
  3917.6      .1       0  3945.4     .16       0  4387.3      .1       0
  4997.1     .07       0  5003.1      .1       0  5066.1     .05       0
  5303.3      .1       0  6002.8     .05       0  6146.2      .1       0
  6485.8     .05       0  6544.1      .1       0  6637.6     .05       0
Bank Sta=4947.3,5049.5
XS Rating Curve= 0 ,0
Exp/Cntr=0.3,0.1

Type RM Length L Ch R = 1 ,113468  ,841,841,841
BEGIN DESCRIPTION:
NORTH GRAPE CREEK 150.0
END DESCRIPTION:
XS GIS Cut Line= 3
      2810943.48     10091290.72      2812401.78     10090223.04
      2812636.15     10089719.58
#Sta/Elev= 30
  3459.8 1725.32  3511.6 1724.89  3547.2 1723.19  3553.4 1721.77  3582.7 1723.23
  3603.5 1721.11  3662.2 1719.71  3747.9  1714.8  3774.9 1714.73  3812.7 1704.65
  3833.6 1701.28  3869.1 1704.98  3912.1 1701.78  4176.4 1699.32  4705.3 1698.24
  4816.2 1699.27  4870.4 1699.48  4956.1 1696.59  4964.6  1696.5  4988.6 1691.88
  4991.4 1691.38  4994.6 1691.88  5014.8 1692.64  5035.6 1701.05  5306.6 1711.19
  5505.3  1721.6  5557.1 1724.99  5635.7 1734.27  5751.7 1752.64  5822.5 1758.79
#Mann= 9 ,-1 , 0
  3459.8     .16       0  3774.9      .1       0  4816.2     .16       0
  4956.1      .1       0  4988.6     .04       0  4994.6      .1       0
  5306.6      .1       0  5505.3     .16       0  5635.7      .1       0
#XS Ineff= 2 , 0
         3870.46 1705.03
Permanent Ineff=
       F       F
Bank Sta=4870.4,5035.6
XS Rating Curve= 0 ,0
Exp/Cntr=0.3,0.1

Type RM Length L Ch R = 1 ,112627  ,1047,1047,1047
BEGIN DESCRIPTION:
NORTH GRAPE CREEK 149.0
END DESCRIPTION:
XS GIS Cut Line= 3
      2811056.34     10091438.29      2812610.11     10090795.95
      2813009.43     10090101.49
#Sta/Elev= 30
  3944.8 1726.92  4120.2 1724.65  4363.1 1718.69  4488.9 1709.12  4509.8 1707.94
  4522.8 1705.52  4535.5 1704.64  4783.5 1701.05    4921 1700.89  4953.4 1699.84
  4967.1 1700.87  4975.1 1695.22  4985.6 1690.78  4993.7 1688.92  4996.5 1688.42
  4999.7 1688.92  5029.2 1692.64  5061.7 1693.23  5104.9 1696.03  5153.7 1696.49
  5234.8  1695.4  5464.6 1697.25  5475.4 1696.56  5676.8 1695.39  5757.3 1698.96
  5928.3 1703.16    6066 1708.55  6155.7 1712.54  6336.5 1720.32  6427.2 1725.65
#Mann= 9 ,-1 , 0
  3944.8      .1       0  4488.9     .16       0  4535.5      .1       0
  4993.7     .07       0  4999.7      .1       0  5153.7     .16       0
  5475.4      .1       0    6066     .05       0  6155.7      .1       0
#XS Ineff= 2 , 0
         4966.05 1700.88
Permanent Ineff=
       F       F
Bank Sta=4975.1,5104.9
XS Rating Curve= 0 ,0
Exp/Cntr=0.3,0.1

Type RM Length L Ch R = 1 ,111580  ,502,502,502
BEGIN DESCRIPTION:
NORTH GRAPE CREEK 148.0
END DESCRIPTION:
XS GIS Cut Line= 4
      2811169.12     10091811.58      2813000.74     10091203.94
      2813226.43     10091065.05      2813269.79     10090067.78
#Sta/Elev= 30
  3241.5 1730.72  3265.2 1730.87  3365.8 1728.46  3509.7 1723.03    3578 1722.26
  3646.8  1718.5  3758.6 1713.89  3898.1 1706.54  4011.7 1704.48  4515.6 1694.77
  4679.3 1693.45  4768.5 1695.23  4800.1 1693.07  4958.2 1692.11  4979.2 1689.96
  4998.4  1682.7  5001.2  1682.2  5004.4  1682.7  5027.8 1688.24    5053 1687.04
  5096.5 1690.31    5205 1692.65  5275.8 1692.86  5443.9 1689.12  5887.6 1703.46
  6034.2 1708.88  6238.4 1719.63  6323.3 1726.68  6378.5 1731.95  6434.5 1734.22
#Mann= 15 ,-1 , 0
  3241.5      .1       0  3265.2     .05       0  3365.8      .1       0
  3509.7     .05       0  3646.8      .1       0  3758.6     .16       0
  3898.1     .05       0  4011.7      .1       0  4998.4     .07       0
  5004.4      .1       0  5275.8     .16       0  5443.9      .1       0
  5887.6     .05       0  6034.2      .1       0  6323.3     .05       0
#XS Ineff= 2 , 0
          4766.9 1695.21 5249.93         1693.54
Permanent Ineff=
       F       F
Bank Sta=4958.2,5205
XS Rating Curve= 0 ,0
Exp/Cntr=0.3,0.1

Type RM Length L Ch R = 1 ,111078  ,991,991,991
BEGIN DESCRIPTION:
Mapping XS 980993ad
END DESCRIPTION:
XS GIS Cut Line= 4
      2811446.78     10092077.06      2813287.01     10091643.04
      2813399.86     10091226.37      2813399.86     10090280.17
#Sta/Elev= 30
  3427.7 1723.58  3457.9 1721.95  3612.6 1716.16  3765.2 1710.89  4058.5 1699.52
  4226.3 1696.03  4417.2 1695.47  4584.7 1692.71  4643.6 1686.76  4680.8 1692.77
    4892 1690.61  4908.9  1689.9  4970.6 1686.11  4998.4 1681.64  5001.2 1681.14
  5004.4 1681.64  5029.7 1686.85  5061.9 1688.64    5072 1690.31  5199.3 1690.89
  5268.2 1690.82    5442 1690.67  5597.4 1686.28  5734.6  1691.2  5822.7 1695.83
  5898.7 1696.25  6252.7 1700.99  6430.5 1707.89    6533 1711.94  6696.3 1720.18
#Mann= 18 ,-1 , 0
  3427.7      .1       0  3457.9     .16       0  3612.6      .1       0
  3765.2     .05       0  4058.5      .1       0  4226.3     .05       0
  4417.2      .1       0  4584.7     .16       0    4892      .1       0
  4998.4     .07       0  5004.4      .1       0  5061.9     .16       0
  5199.3     .05       0  5268.2      .1       0  5734.6     .16       0
  5898.7      .1       0  6430.5     .05       0    6533      .1       0
#XS Ineff= 2 , 0
         4714.25 1693.07
Permanent Ineff=
       F       F
Bank Sta=4908.9,5072
XS Rating Curve= 0 ,0
Exp/Cntr=0.3,0.1
