HEC-RAS study NORTH GRAPE CREEK.prj: NORTH GRAPE CREEK Base Level Engineering

--- NORTH GRAPE CREEK.g01 (geometry) --- (continued)

Type RM Length L Ch R = 1 ,63092   ,1010,1010,1010
BEGIN DESCRIPTION:
NORTH GRAPE CREEK 81.0
END DESCRIPTION:
XS GIS Cut Line= 2
      2844728.02     10096186.86      2843226.44     10096062.76
#Sta/Elev= 30
  4338.5 1491.33  4435.3 1489.35  4488.6 1486.81    4619 1483.08  4719.3 1478.08
  4789.6  1472.8  4806.4 1470.64  4839.8 1464.77  4859.8 1457.95  4869.9 1454.19
  4879.9 1452.26    4923 1451.32  4984.9 1451.32  5077.6 1450.23  5080.3 1449.73
  5083.6 1450.23  5102.4 1450.45  5130.7 1452.97  5150.8 1456.78  5160.7 1459.71
  5170.9 1461.62  5214.9 1466.33  5251.2 1469.44  5286.7 1474.24  5311.4 1475.72
  5451.8 1480.87  5533.5 1485.67  5649.4 1490.25  5817.2 1495.32  5845.2 1495.74
#Mann= 9 ,-1 , 0
  4338.5      .1       0  4806.4     .05       0    4923     .16       0
  4984.9     .05       0  5077.6    .035       0  5083.6     .05       0
  5102.4     .16       0  5214.9      .1       0  5817.2     .16       0
Bank Sta=4859.8,5160.7
XS Rating Curve= 0 ,0
Exp/Cntr=0.3,0.1

Type RM Length L Ch R = 1 ,62082   ,1081,1081,1081
BEGIN DESCRIPTION:
NORTH GRAPE CREEK 80.0
END DESCRIPTION:
XS GIS Cut Line= 3
      2845050.63     10096137.21      2844380.53     10095119.66
      2843834.52     10094734.97
#Sta/Elev= 30
  4106.1 1491.52  4385.7 1482.29  4578.5 1472.18  4601.2 1469.06  4738.1 1459.45
  4753.2 1456.22  4816.7  1449.6  4831.4 1446.65  4882.7 1443.48  5048.3 1443.58
  5096.5 1442.45  5099.3 1441.95  5102.5 1442.45  5135.7 1443.34  5157.8 1448.88
  5163.9 1451.29  5250.1 1473.86  5281.6 1478.84  5344.4 1486.31  5380.1 1488.71
  5582.2 1495.36  5754.6 1503.77  5881.8 1517.15  5882.5 1517.16  5897.4 1519.85
  5918.4 1520.73  5933.1 1523.38  5968.9  1525.7  5983.7  1528.4  5992.4 1528.03
#Mann= 7 ,-1 , 0
  4106.1      .1       0  5096.5     .07       0  5102.5      .1       0
  5157.8     .16       0  5281.6      .1       0  5881.8     .05       0
  5882.5      .1       0
Bank Sta=4816.7,5163.9
XS Rating Curve= 0 ,0
Exp/Cntr=0.3,0.1

Type RM Length L Ch R = 1 ,61001   ,645,645,645
BEGIN DESCRIPTION:
NORTH GRAPE CREEK 79.0
END DESCRIPTION:
XS GIS Cut Line= 3
      2845433.45     10095851.96      2845530.96     10095183.32
       2845043.4     10094180.35
#Sta/Elev= 30
  4216.7  1477.6  4457.4 1470.25  4548.4 1465.22  4568.6 1463.09  4703.5 1457.73
  4730.3 1454.87  4773.5 1452.75  4838.5  1443.6  4853.9 1443.08    4895 1440.72
  4954.2 1433.27  4983.7 1432.61    4989 1432.52  4991.8 1432.02    4995 1432.52
  5028.1 1434.15  5140.2 1435.12  5224.9 1434.16  5290.1 1437.17  5320.6 1442.34
  5371.3 1448.95  5416.4 1452.15  5425.7 1451.83  5492.4 1458.91  5725.9 1477.67
  5777.3 1485.18    5800 1486.59  5895.7 1494.91  5912.6 1497.33  6007.6 1503.28
#Mann= 8 ,-1 , 0
  4216.7     .16       0  4853.9      .1       0  4983.7     .16       0
    4989     .07       0    4995     .16       0  5028.1      .1       0
  5290.1     .16       0    5800      .1       0
Bank Sta=4895,5320.6
XS Rating Curve= 0 ,0
Exp/Cntr=0.3,0.1

Type RM Length L Ch R = 1 ,60356   ,591,591,591
BEGIN DESCRIPTION:
NORTH GRAPE CREEK 78.0
END DESCRIPTION:
XS GIS Cut Line= 3
      2846561.79     10095169.36      2846088.18     10094751.47
       2845212.2     10094139.67
#Sta/Elev= 30
  4145.5  1476.3  4222.7 1468.29  4286.2 1463.27  4371.6 1459.48  4420.9 1454.24
  4512.9 1448.65  4612.5  1445.6  4676.1 1441.31  4690.3 1442.05  4768.1 1437.99
  4825.6 1436.75  4883.4 1433.53  4940.3 1429.86  5002.7 1428.24  5005.4 1427.74
  5008.7 1428.24  5077.2 1430.56  5164.7 1428.72  5184.5 1430.09  5205.4 1429.13
  5228.1 1430.16  5276.9 1436.71  5537.8 1465.41  5565.7  1468.8    5594 1474.85
  5672.9 1487.93  5687.8 1488.69  5759.3  1497.2  5765.4 1498.84  5845.6 1506.92
#Mann= 6 ,-1 , 0
  4145.5     .16       0  4883.4      .1       0  5002.7     .07       0
  5008.7      .1       0  5164.7     .16       0  5537.8      .1       0
Bank Sta=4825.6,5276.9
XS Rating Curve= 0 ,0
Exp/Cntr=0.3,0.1

Type RM Length L Ch R = 1 ,59765   ,729,729,729
BEGIN DESCRIPTION:
NORTH GRAPE CREEK 77.0
END DESCRIPTION:
XS GIS Cut Line= 2
      2846882.23     10094695.75      2845503.25      10093762.5
#Sta/Elev= 30
  4067.5  1481.3  4256.8 1468.36  4345.7 1461.97  4459.6 1458.95  4669.4 1448.04
  4834.1 1431.31  4899.4 1425.48  4989.9 1423.83  4992.6 1423.33  4995.9 1423.83
  5006.8 1424.02  5145.6 1425.31  5166.6  1427.9  5187.6 1433.48  5253.5 1437.34
  5295.5  1443.2  5310.4  1447.2  5331.4 1447.98  5346.4 1451.68  5372.5 1452.58
  5382.3 1455.17  5403.3 1455.06  5412.2 1457.04  5418.3 1455.23  5433.2 1459.35
  5454.2  1458.5  5505.1 1471.65    5628 1488.74  5691.1  1494.4  5732.6 1496.99
#Mann= 9 ,-1 , 0
  4067.5      .1       0  4256.8     .16       0  4669.4      .1       0
  4899.4     .16       0  4989.9     .07       0  4995.9     .16       0
  5006.8      .1       0  5372.5     .16       0  5691.1     .05       0
Bank Sta=4834.1,5187.6
XS Rating Curve= 0 ,0
Exp/Cntr=0.3,0.1

Type RM Length L Ch R = 1 ,59036   ,710,710,710
BEGIN DESCRIPTION:
NORTH GRAPE CREEK 76.0
END DESCRIPTION:
XS GIS Cut Line= 2
      2847174.75     10094347.45      2845712.75     10092704.45
#Sta/Elev= 30
  4207.9 1497.18  4210.3  1496.9  4399.5 1487.65    4555 1473.74  4575.9 1470.74
  4618.3 1467.81  4753.2 1454.65  4824.3 1445.18    4872 1436.75  4895.3 1432.11
  4908.9 1427.78  4930.5 1418.56  4941.7 1417.44  4944.4 1416.94  4947.7 1417.44
  5036.7 1417.81  5128.6 1419.99  5149.9 1423.26  5161.2 1423.77  5234.8 1425.06
  5302.5 1430.17  5348.5 1433.21  5440.9 1435.71  5483.2 1436.58  5581.8 1442.17
  5681.3 1443.65  5808.4 1450.32  6120.3 1479.98  6317.9 1492.09  6407.2 1494.98
#Mann= 10 ,-1 , 0
  4207.9     .16       0  4210.3      .1       0  4618.3     .16       0
    4872      .1       0  4941.7     .07       0  4947.7      .1       0
  5161.2     .16       0  5302.5      .1       0  5440.9     .16       0
  6317.9      .1       0
Bank Sta=4908.9,5149.9
XS Rating Curve= 0 ,0
Exp/Cntr=0.3,0.1

Type RM Length L Ch R = 1 ,58326   ,852,852,852
BEGIN DESCRIPTION:
NORTH GRAPE CREEK 75.0
END DESCRIPTION:
XS GIS Cut Line= 2
       2847773.8     10093623.09      2846032.93     10092606.42
#Sta/Elev= 30
  4097.6 1494.14  4364.2 1481.47  4486.3 1470.93  4596.7 1464.47  4597.6  1464.4
  4671.2 1457.93  4800.6 1441.45  4839.5 1436.42  4868.1 1428.93  4882.5 1421.59
  4891.2 1417.06  4898.2 1415.35  5039.9 1413.93  5042.7 1413.43  5045.9 1413.93
  5089.3 1414.32  5111.3 1415.04    5146 1421.12    5176 1425.61  5234.7 1430.37
  5395.1 1436.61  5400.9 1437.99  5521.1 1444.13  5670.9  1449.5  5694.3 1451.52
  5704.3 1454.03  5737.3 1460.82  5881.5 1470.13  5906.3 1471.78  6113.6 1484.43
#Mann= 13 ,-1 , 0
  4097.6      .1       0  4486.3     .16       0  4596.7      .1       0
  4597.6     .16       0  4800.6      .1       0  5039.9     .07       0
  5045.9      .1       0  5089.3     .16       0  5521.1      .1       0
  5670.9     .16       0  5704.3      .1       0  5881.5     .16       0
  5906.3      .1       0
Bank Sta=4882.5,5146
XS Rating Curve= 0 ,0
Exp/Cntr=0.3,0.1

Type RM Length L Ch R = 1 ,57474   ,593,593,593
BEGIN DESCRIPTION:
NORTH GRAPE CREEK 74.0
END DESCRIPTION:
XS GIS Cut Line= 3
      2848261.37      10092898.7      2847564.83     10092452.91
      2846382.05      10092258.1
#Sta/Elev= 30
  3960.1 1475.96  4089.1 1473.75  4270.9 1467.34  4343.5 1462.33    4407 1455.46
  4552.5 1446.31  4631.1 1436.95  4711.6  1429.6  4740.2 1424.91    4782 1415.17
  4787.1 1415.17  4823.9 1408.82  4844.2 1407.12  4962.8 1405.44  4965.6 1404.94
  4968.8 1405.44  5077.3 1407.23  5121.7 1410.01  5133.7 1412.26  5148.2 1414.93
  5209.1 1421.87    5239 1422.88  5298.4 1427.79  5330.7 1429.21  5411.8 1436.26
  5488.5 1449.03  5533.4    1453    5582 1454.93  5664.8 1458.11  5985.8 1471.43
#Mann= 9 ,-1 , 0
  3960.1     .16       0  4711.6      .1       0  4962.8     .07       0
  4968.8      .1       0  5133.7     .16       0  5298.4      .1       0
  5488.5     .16       0    5582      .1       0  5664.8     .16       0
Bank Sta=4787.1,5148.2
XS Rating Curve= 0 ,0
Exp/Cntr=0.3,0.1

Type RM Length L Ch R = 1 ,56881   ,548,548,548
BEGIN DESCRIPTION:
NORTH GRAPE CREEK 73.0
END DESCRIPTION:
XS GIS Cut Line= 3
      2848526.03     10092661.85      2847509.11     10091798.17
      2847286.23     10091143.46
#Sta/Elev= 30
  3953.7 1466.38  4220.3 1460.84  4404.8 1454.54  4454.2 1448.93  4539.9 1445.42
  4603.6 1439.29  4638.8 1434.86  4710.2 1422.91  4780.4 1408.73  4866.1 1405.84
  4929.8 1400.17  4950.7  1400.8    4984 1399.34  4986.7 1398.84    4990 1399.34
    5042 1399.97  5064.9 1400.12  5074.2 1401.97  5114.4 1405.53  5142.9 1408.56
  5170.7  1418.6  5184.6 1421.79  5241.8 1429.36  5463.7 1439.68  5552.5 1449.31
  5620.5 1454.03  5725.7 1466.51  5801.1 1471.25  5833.9 1473.09  5979.5 1476.41
#Mann= 7 ,-1 , 0
  3953.7     .16       0    4984     .07       0    4990     .16       0
    5042      .1       0  5074.2     .16       0  5801.1      .1       0
  5833.9     .16       0
Bank Sta=4866.1,5114.4
XS Rating Curve= 0 ,0
Exp/Cntr=0.3,0.1

Type RM Length L Ch R = 1 ,56333   ,686,686,686
BEGIN DESCRIPTION:
NORTH GRAPE CREEK 72.0
END DESCRIPTION:
XS GIS Cut Line= 2
      2848539.99     10092174.31      2847759.88     10091129.52
#Sta/Elev= 30
  4305.8 1451.05  4429.4 1447.01  4485.7 1447.33  4543.6 1444.59  4593.6 1439.21
  4629.5 1434.11  4650.4 1429.63  4685.8 1425.15    4715  1417.4  4735.8 1408.67
  4750.4 1404.37  4771.3  1403.5    4815 1405.85  4851.5 1404.73  4865.1 1403.99
  4893.1 1399.38  4903.8 1399.05  4906.5 1398.55  4909.8 1399.05  5029.8 1399.22
  5050.6 1402.92  5105.1 1405.63  5150.7 1404.51  5206.9 1420.44  5236.1 1426.88
  5346.5  1447.3  5371.6 1451.09    5484 1462.46  5507.4 1464.76  5609.7 1472.81
#Mann= 8 ,-1 , 0
  4305.8     .16       0  4851.5     .05       0  4903.8    .033       0
  4909.8     .05       0  5105.1     .16       0  5346.5      .1       0
    5484     .16       0  5507.4      .1       0
Bank Sta=4865.1,5050.6
XS Rating Curve= 0 ,0
Exp/Cntr=0.3,0.1

Type RM Length L Ch R = 1 ,55647   ,687,687,687
BEGIN DESCRIPTION:
NORTH GRAPE CREEK 71.0
END DESCRIPTION:
XS GIS Cut Line= 4
      2848762.87     10092090.75      2848707.14     10091422.04
      2848470.32     10090934.47      2848359.01     10090628.35
#Sta/Elev= 30
  4166.5 1454.56  4263.9 1451.38  4394.3 1441.68  4685.3 1401.66  4735.5 1400.33
  4775.6 1402.11  4815.8  1400.7  4871.7 1396.58  4921.6 1395.69  4924.3 1395.19
  4927.6 1395.69  4946.8 1396.93  5001.5 1395.97  5035.8 1396.78  5074.8 1401.85
  5113.6    1404  5135.8 1406.94  5170.6  1414.8  5277.8 1431.61  5305.9 1434.45
  5377.2 1446.89  5453.8 1455.73  5497.4 1463.53  5520.3 1465.38    5540 1468.88
  5625.1 1478.54  5632.1 1480.37  5637.4 1479.93  5693.3 1486.22  5705.3 1488.76
#Mann= 3 ,-1 , 0
  4166.5     .16       0  4921.6     .07       0  4927.6     .16       0
Bank Sta=4815.8,5074.8
XS Rating Curve= 0 ,0
Exp/Cntr=0.3,0.1

Type RM Length L Ch R = 1 ,54960   ,879,879,879
BEGIN DESCRIPTION:
NORTH GRAPE CREEK 70.0
END DESCRIPTION:
XS GIS Cut Line= 2
       2849278.3     10092188.19       2849278.3     10090488.69
#Sta/Elev= 30
  3914.2 1457.17  3978.7 1452.74  4028.7 1446.17  4138.7 1437.57  4158.7 1434.81
  4248.7  1428.3  4358.7 1423.47  4528.7 1413.63  4648.7 1409.75  4688.7 1407.16
  4718.7 1403.71  4752.2 1402.44  4788.7 1398.78  4878.7 1395.15  4909.8 1391.78
  4948.7 1388.33  5045.7 1387.77  5048.4 1387.27  5051.7 1387.77  5098.7 1389.58
  5108.7 1394.42  5138.7 1419.62  5158.7 1425.42  5228.7 1438.48  5268.7 1447.33
  5348.7 1461.26  5458.7 1478.19  5558.7 1488.91  5598.7 1491.93  5613.7  1494.3
#Mann= 5 ,-1 , 0
  3914.2     .16       0  4752.2      .1       0  4909.8     .16       0
  5045.7     .07       0  5051.7     .16       0
Bank Sta=4878.7,5108.7
XS Rating Curve= 0 ,0
Exp/Cntr=0.3,0.1

Type RM Length L Ch R = 1 ,54081   ,567,567,567
BEGIN DESCRIPTION:
NORTH GRAPE CREEK 69.0
END DESCRIPTION:
XS GIS Cut Line= 3
      2849626.58     10092355.36      2850058.42     10091380.25
      2850030.56     10090669.75
#Sta/Elev= 30
  3722.3 1452.71  3838.5 1444.46  4105.6    1432  4172.5 1427.21  4331.5 1420.25
  4539.9 1413.83  4577.9 1412.21  4754.7 1403.48  4895.4 1388.74  4917.1 1386.64
  4955.4 1380.84  5012.4 1378.56  5015.2 1378.06  5018.4 1378.56  5105.5 1379.25
  5115.5 1381.05  5125.5 1388.41  5135.5 1397.04  5140.5 1405.71  5145.5 1414.38
  5155.6 1422.96  5170.4 1425.31  5175.6 1428.39  5225.6 1439.04  5295.7 1449.99
  5355.7 1456.63  5395.7 1459.35  5423.1 1463.98  5428.1 1463.07  5499.8 1468.15
#Mann= 7 ,-1 , 0
  3722.3     .16       0  4539.9      .1       0  4577.9     .16       0
  4917.1      .1       0  5012.4     .07       0  5018.4      .1       0
  5140.5     .16       0
Bank Sta=4895.4,5125.5
XS Rating Curve= 0 ,0
Exp/Cntr=0.3,0.1

Type RM Length L Ch R = 1 ,53514   ,774,774,774
BEGIN DESCRIPTION:
NORTH GRAPE CREEK 68.0
END DESCRIPTION:
XS GIS Cut Line= 3
      2850518.13     10092536.49      2850601.71     10091045.91
      2850267.74     10090377.97
#Sta/Elev= 30
  3765.3 1439.32  3928.3 1436.34  3998.4 1431.06  4098.6 1427.02  4419.1 1420.04
  4739.6 1402.78  4839.7 1393.92  4909.9 1384.15  4933.6 1380.45  4949.9 1375.64
  4981.3 1373.19    4997 1372.81  4999.7 1372.31    5003 1372.81  5070.1 1374.98
  5113.6 1382.01  5130.2 1385.81  5180.3 1399.99  5200.3 1403.77  5256.8  1412.3
  5316.2 1417.79  5362.9 1426.06  5433.6 1433.88  5517.4 1438.44  5612.5 1448.65
  5668.4 1451.41  5812.3 1459.59  5902.3 1462.55  6003.4  1466.3    6005 1466.27
#Mann= 10 ,-1 , 0
  3765.3     .16       0  4981.3      .1       0    4997     .07       0
    5003      .1       0  5113.6     .16       0  5362.9      .1       0
  5668.4     .16       0  5812.3      .1       0  5902.3     .16       0
  6003.4      .1       0
Bank Sta=4909.9,5130.2
XS Rating Curve= 0 ,0
Exp/Cntr=0.3,0.1

Type RM Length L Ch R = 1 ,52740   ,687,687,687
BEGIN DESCRIPTION:
NORTH GRAPE CREEK 67.0
END DESCRIPTION:
XS GIS Cut Line= 3
      2850991.77     10092829.05      2851158.94     10091770.31
      2851827.63     10090920.51
#Sta/Elev= 30
  3732.7 1442.69  3873.3 1437.93    4143 1423.91  4325.5 1411.08  4382.9  1403.2
  4450.3 1400.19    4467 1396.96  4512.8 1396.59  4517.8 1399.86  4580.3 1400.19
  4760.6 1392.88  4923.1  1377.8  4972.8 1369.65  4998.7 1368.72  5001.4 1368.22
  5004.7 1368.72  5041.1 1369.54  5065.8 1371.62    5093 1378.52  5102.9 1386.14
  5107.5 1388.73  5115.5  1399.8    5130 1410.77  5150.8 1416.83  5200.5 1423.04
  5295.5 1428.95  5421.9 1437.16  5542.1 1449.37  5599.9 1451.38  5885.9 1471.42
#Mann= 6 ,-1 , 0
  3732.7     .16       0  4998.7     .07       0  5004.7     .16       0
  5041.1      .1       0  5102.9     .16       0  5295.5      .1       0
#XS Ineff= 2 , 0
         4580.51 1400.24
Permanent Ineff=
       F       F
Bank Sta=4923.1,5093
XS Rating Curve= 0 ,0
Exp/Cntr=0.3,0.1

Type RM Length L Ch R = 1 ,52053   ,709,709,709
BEGIN DESCRIPTION:
NORTH GRAPE CREEK 66.0
END DESCRIPTION:
XS GIS Cut Line= 2
      2851493.28     10092968.33      2852175.29     10091117.17
#Sta/Elev= 30
  3953.6 1443.86  4118.4 1440.05  4203.6 1434.69  4310.2  1424.4  4406.1 1419.74
  4505.5 1408.56  4667.5 1398.44  4779.1 1386.58  4828.4 1384.01  4896.3 1376.58
  4917.6 1371.18  4961.1  1366.3  4993.5 1365.94  4996.3 1365.44  4999.5 1365.94
  5052.1 1369.21  5082.5 1367.67  5120.1 1378.76  5179.3 1383.25  5184.7 1383.68
    5285 1395.47  5315.5 1401.71  5340.6 1411.19  5345.9 1408.88  5356.4 1411.22
  5431.9 1419.84  5543.1 1438.19  5642.3 1448.47  5801.1 1462.54  5926.4 1468.32
#Mann= 9 ,-1 , 0
  3953.6     .16       0  4667.5      .1       0  4828.4     .16       0
  4961.1      .1       0  4993.5     .07       0  4999.5      .1       0
  5179.3     .16       0  5184.7      .1       0  5356.4     .16       0
Bank Sta=4896.3,5120.1
XS Rating Curve= 0 ,0
Exp/Cntr=0.3,0.1

Type RM Length L Ch R = 1 ,51344   ,1170,1170,1170
BEGIN DESCRIPTION:
NORTH GRAPE CREEK 65.0
END DESCRIPTION:
XS GIS Cut Line= 2
      2852482.35     10093219.13      2852621.54     10090866.74
#Sta/Elev= 30
  3891.3  1448.6    3906 1445.63  4117.1 1430.01  4507.8 1404.25  4537.8 1400.11
  4577.9  1398.2  4728.2 1383.53  4768.2 1375.02  4808.3 1372.71  4830.8 1370.66
  4908.5 1364.91  5038.3    1363  5055.7 1362.53  5058.5 1362.03  5061.7 1362.53
  5091.3 1363.55  5108.8 1364.14  5148.8 1372.02    5189 1383.65    5219 1397.01
  5249.1 1403.08  5349.2 1409.38  5449.4 1425.58  5539.6 1434.93  5619.7 1438.76
  5739.9 1447.94  5877.3 1449.84  5983.3 1447.52  6065.9 1446.95  6247.8 1447.98
#Mann= 10 ,-1 , 0
  3891.3     .16       0  4830.8      .1       0  5038.3     .16       0
  5055.7     .07       0  5061.7     .16       0  5091.3      .1       0
  5148.8     .16       0  5877.3      .1       0  5983.3     .05       0
  6065.9      .1       0
Bank Sta=4808.3,5148.8
XS Rating Curve= 0 ,0
Exp/Cntr=0.3,0.1

Type RM Length L Ch R = 1 ,50174   ,1304,1304,1304
BEGIN DESCRIPTION:
Mapping XS 4f631ae7
END DESCRIPTION:
XS GIS Cut Line= 2
       2853596.8     10093316.66      2853750.04     10091463.88
#Sta/Elev= 30
  3985.9 1443.53  4018.9 1442.74  4119.3 1435.98    4330  1414.8  4368.7 1412.62
  4449.9 1409.68  4580.9 1394.77  4761.5 1380.97  4781.5 1377.93  4801.6 1370.02
  4851.8 1367.16  4891.9 1362.56    4932 1358.16  4952.5 1358.24  4989.2 1355.44
    4992 1354.94  4995.2 1355.44  5030.2 1356.84  5062.5 1357.01  5082.6 1362.78
  5112.7 1365.31  5132.7 1369.15  5158.2 1383.39  5273.2 1413.17  5303.3 1423.48
  5383.6 1438.21  5534.1 1458.54  5614.4 1465.54  5654.5 1470.95    5845 1483.09
#Mann= 7 ,-1 , 0
  3985.9     .16       0  4368.7      .1       0  4449.9     .16       0
  4952.5      .1       0  4989.2     .07       0  4995.2      .1       0
  5030.2     .16       0
Bank Sta=4891.9,5082.6
XS Rating Curve= 0 ,0
Exp/Cntr=0.3,0.1

Type RM Length L Ch R = 1 ,48870   ,1063,1063,1063
BEGIN DESCRIPTION:
NORTH GRAPE CREEK 61.0
END DESCRIPTION:
XS GIS Cut Line= 2
      2854975.94     10093219.05      2854962.01      10091449.9
#Sta/Elev= 30
  4225.4 1397.28  4470.7 1379.73  4655.1 1369.68  4700.7 1365.91  4810.7 1361.33
  4840.7 1362.59  4850.7 1362.52  4880.7 1358.71  4910.7 1357.91  4930.7 1353.22
  4947.7 1353.13  4950.5 1352.63  4953.7 1353.13  5000.7 1353.64  5040.7 1358.07
  5076.1 1359.81  5090.7 1360.82  5120.7 1362.46  5150.7 1370.39  5190.7 1384.63
  5250.7 1396.65  5330.7 1405.43  5410.8 1416.88  5480.8 1421.06  5530.8  1425.5
  5580.8 1428.01  5811.7 1432.19  5890.8 1434.05  5940.8 1433.36  5994.6  1434.2
#Mann= 6 ,-1 , 0
  4225.4     .16       0  4655.1      .1       0  4947.7     .07       0
  4953.7      .1       0  5076.1     .16       0  5811.7      .1       0
Bank Sta=4840.7,5090.7
XS Rating Curve= 0 ,0
Exp/Cntr=0.3,0.1

Type RM Length L Ch R = 1 ,47807   ,979,979,979
BEGIN DESCRIPTION:
NORTH GRAPE CREEK 60.0
END DESCRIPTION:
XS GIS Cut Line= 2
       2855825.7     10093442.03      2856201.44     10091646.83
#Sta/Elev= 30
  4089.2 1414.68  4130.3 1413.06  4262.6 1402.06  4455.3 1383.71  4506.3 1382.71
  4625.9  1372.6  4781.8 1360.44  4874.1 1353.38  4888.1 1352.01  4953.9 1346.36
  5014.2 1345.94  5016.9 1345.44  5020.2 1345.94  5030.9 1346.66  5047.8  1351.9
  5053.8 1356.81  5058.9 1356.65  5078.5 1371.06  5098.6 1383.14  5103.7 1383.09
  5109.1 1387.85  5129.6    1394  5198.5 1408.37  5272.6 1416.09  5303.5 1422.24
  5498.2 1435.39  5587.9 1437.83  5599.5 1439.75  5837.6 1449.04  5923.3 1449.77
#Mann= 8 ,-1 , 0
  4089.2      .1       0  4262.6     .16       0  4625.9      .1       0
  4781.8     .16       0  4888.1      .1       0  5014.2     .07       0
  5020.2      .1       0  5030.9     .16       0
Bank Sta=4874.1,5053.8
XS Rating Curve= 0 ,0
Exp/Cntr=0.3,0.1

Type RM Length L Ch R = 1 ,46828   ,1011,1011,1011
BEGIN DESCRIPTION:
NORTH GRAPE CREEK 59.0
END DESCRIPTION:
XS GIS Cut Line= 2
      2856550.09     10093539.52      2857204.14     10092412.33
#Sta/Elev= 30
  4232.4 1403.36  4322.3 1398.33  4375.3 1390.85  4412.5 1387.24  4439.9 1381.58
  4482.9 1376.99  4573.2 1371.97  4600.5 1369.01  4637.8 1368.08  4676.3 1365.43
  4716.8  1364.2  4819.9 1359.43  4857.2  1356.4    4873 1352.14    4916 1344.98
  4944.3  1343.6  5014.8 1343.37  5017.6 1342.87  5020.8 1343.37  5092.4 1345.28
  5106.2 1347.75  5113.9 1351.62  5135.4 1358.97    5157  1364.7  5172.7 1375.52
  5194.2  1384.5  5229.5    1390  5354.9  1407.2    5494 1418.21  5535.6 1419.47
#Mann= 6 ,-1 , 0
  4232.4      .1       0  4676.3     .16       0  4716.8      .1       0
  5014.8     .07       0  5020.8      .1       0  5229.5     .16       0
Bank Sta=4857.2,5113.9
XS Rating Curve= 0 ,0
Exp/Cntr=0.3,0.1

Type RM Length L Ch R = 1 ,45817   ,802,802,802
BEGIN DESCRIPTION:
NORTH GRAPE CREEK 58.0
END DESCRIPTION:
XS GIS Cut Line= 3
       2856954.1     10093776.31      2857734.21     10093372.33
      2858333.19     10092898.72
#Sta/Elev= 30
    3982 1399.15  4061.9 1395.21  4084.1 1392.11  4211.2 1384.34  4233.4  1381.4
    4344 1376.03  4426.1 1367.39  4484.5 1364.78  4758.5 1352.17  4847.5 1346.08
  4877.4 1342.81    4927 1342.75  5002.6 1338.82  5005.3 1338.32  5008.6 1338.82
  5034.6 1342.19  5069.7  1342.9  5090.5 1349.95  5096.9 1355.27  5133.6 1371.12
  5146.6 1374.41  5175.5  1377.6  5218.8 1385.77    5254 1388.33  5297.3 1394.42
  5353.4 1395.77  5375.9  1400.2  5422.5 1404.57  5601.8 1417.95  5624.1 1418.79
#Mann= 8 ,-1 , 0
    3982      .1       0  4484.5     .16       0  4758.5      .1       0
  5002.6     .07       0  5008.6      .1       0  5034.6     .16       0
  5422.5      .1       0  5601.8     .05       0
Bank Sta=4847.5,5090.5
XS Rating Curve= 0 ,0
Exp/Cntr=0.3,0.1

Type RM Length L Ch R = 1 ,45015   ,1195,1195,1195
BEGIN DESCRIPTION:
NORTH GRAPE CREEK 54.0
END DESCRIPTION:
XS GIS Cut Line= 2
      2857176.94     10094194.25      2859071.57     10093664.87
#Sta/Elev= 30
  3754.9 1405.21  3813.1 1403.83  3920.7 1394.95  4119.9 1387.57  4234.1 1378.92
  4431.4 1368.59  4686.3  1357.2  4732.4 1353.67  4790.1 1350.23  4821.6 1347.49
  4852.5 1342.76  4919.4 1340.33  4989.1 1334.23  4991.8 1333.73  4995.1 1334.23
  5064.7 1337.07  5077.5 1341.88  5085.5 1352.63  5101.2  1364.8  5112.3 1374.26
  5117.5 1374.37  5158.2 1391.27  5185.8 1400.86  5204.9 1402.89  5298.7 1414.98
  5417.8 1425.52    5485 1428.58    5516 1432.85  5689.8 1445.78  5722.1 1447.12
#Mann= 12 ,-1 , 0
  3754.9      .1       0  4686.3     .16       0  4732.4      .1       0
  4790.1     .16       0  4821.6      .1       0  4989.1     .07       0
  4995.1      .1       0  5077.5     .16       0  5101.2      .1       0
  5204.9     .16       0    5516      .1       0  5689.8     .16       0
Bank Sta=4919.4,5077.5
XS Rating Curve= 0 ,0
Exp/Cntr=0.3,0.1

Type RM Length L Ch R = 1 ,43820   ,989,989,989
BEGIN DESCRIPTION:
NORTH GRAPE CREEK 53.0
END DESCRIPTION:
XS GIS Cut Line= 3
      2857037.67     10094709.68      2858402.88     10095002.22
      2858944.84     10094946.63
#Sta/Elev= 30
  3821.6 1412.49  3934.9 1406.71  4054.1 1385.22  4077.8 1383.84  4114.7 1381.94
  4170.1 1376.19  4340.5  1370.7  4374.7 1366.34  4395.1 1360.13  4467.9 1355.01
  4610.3  1350.7    4794 1346.88  4838.4 1340.47  4906.5 1333.75  4918.3 1330.16
  4968.4 1329.44  5036.4 1328.78  5039.2 1328.28  5042.4 1328.78  5061.5 1329.43
  5080.3 1334.39  5107.6 1339.48  5131.5 1351.54  5150.1 1370.87  5155.2 1371.05
  5162.2 1377.18  5199.6 1385.16  5354.6 1400.62  5504.9 1405.95  5762.6 1428.91
#Mann= 10 ,-1 , 0
  3821.6      .1       0  4077.8     .16       0  4114.7      .1       0
  4467.9     .16       0  4610.3      .1       0  4838.4     .16       0
  4968.4     .05       0  5036.4    .033       0  5042.4     .05       0
  5107.6     .16       0
Bank Sta=4906.5,5080.3
XS Rating Curve= 0 ,0
Exp/Cntr=0.3,0.1

Type RM Length L Ch R = 1 ,42831   ,1224,1224,1224
BEGIN DESCRIPTION:
NORTH GRAPE CREEK 52.0
END DESCRIPTION:
XS GIS Cut Line= 3
      2856550.11     10095865.92       2858096.4     10095740.54
      2858848.65     10095420.14
#Sta/Elev= 30
  3828.6 1436.48  3906.4 1433.02  3965.3 1430.98    4158 1422.56  4338.6 1403.84
    4459  1398.1  4509.2 1392.39  4629.6 1366.23  4657.3 1346.93  4679.7 1337.57
  4719.9 1324.87    4747 1322.49  4749.7 1321.99    4753 1322.49  4810.2    1328
  4967.1 1328.36    5051 1327.21  5191.4 1329.91  5241.6 1331.87  5271.7 1337.63
  5321.8 1343.84  5594.3 1351.53  5707.7 1355.07    5844 1362.45  5896.7 1369.86
  5925.3 1379.79  5996.7 1392.35    6067 1399.35  6110.4 1406.54  6197.6 1412.36
#Mann= 9 ,-1 , 0
  3828.6     .16       0  3906.4      .1       0  3965.3     .16       0
    4747     .07       0    4753     .16       0  4967.1      .1       0
  5594.3     .16       0  5707.7      .1       0  5925.3     .16       0
Bank Sta=4679.7,5271.7
XS Rating Curve= 0 ,0
Exp/Cntr=0.3,0.1

Type RM Length L Ch R = 1 ,41607   ,679,679,679
BEGIN DESCRIPTION:
NORTH GRAPE CREEK 50.0
END DESCRIPTION:
XS GIS Cut Line= 3
      2857093.35      10096813.2      2857915.31     10096952.51
      2859182.09     10095978.06
#Sta/Elev= 30
  3954.6 1435.56  4030.8 1428.53  4061.2 1423.86  4107.1 1411.94  4172.8 1403.87
  4283.1 1396.38  4403.8    1383  4456.8 1379.87  4524.5 1360.38  4584.9 1346.66
  4760.7 1337.42  4796.5 1336.51  4846.4 1330.25  4925.2  1315.6  4957.4 1314.61
  4978.5 1314.09  4981.3 1313.59  4984.5 1314.09  5040.5 1316.95  5060.2 1316.37
  5103.7    1329  5153.6 1336.16  5368.1 1340.92  5455.8 1344.16  5795.1 1354.21
    6038 1365.59  6073.3 1369.93  6237.3 1381.06    6337 1400.88  6386.5 1406.48
#Mann= 8 ,-1 , 0
  3954.6      .1       0  4760.7     .16       0  4957.4      .1       0
  4978.5     .07       0  4984.5      .1       0  5040.5     .16       0
  5368.1      .1       0  5455.8     .16       0
Bank Sta=4846.4,5103.7
XS Rating Curve= 0 ,0
Exp/Cntr=0.3,0.1

Type RM Length L Ch R = 1 ,40928   ,1329,1329,1329
BEGIN DESCRIPTION:
NORTH GRAPE CREEK 49.0
END DESCRIPTION:
XS GIS Cut Line= 3
      2857385.95     10098317.71      2858709.35     10097161.47
      2859724.89      10096340.7
#Sta/Elev= 30
  3592.3 1421.68  3675.3 1420.33  3915.1  1409.6  4362.5 1374.94  4411.9 1374.36
  4468.8 1368.11  4645.4 1360.17  4673.9 1355.71  4681.5 1352.15  4702.4  1351.1
  4709.9 1346.59  4724.2 1343.56  4862.3 1324.69  4872.3 1322.68  4944.4 1316.17
    5004 1313.88  5006.8 1313.38    5010 1313.88  5078.2 1315.89  5149.3  1323.1
  5227.1  1328.4  5405.2 1333.36  5503.8  1338.8  5729.8 1345.96  5951.8 1352.38
  6043.7 1355.85  6243.5 1383.91  6371.4  1397.9  6548.9 1410.47  6655.4 1414.51
#Mann= 11 ,-1 , 0
  3592.3     .16       0  3915.1      .1       0  4862.3     .16       0
  4944.4      .1       0    5004     .07       0    5010      .1       0
  5227.1     .16       0  5405.2      .1       0  5503.8     .16       0
  5729.8      .1       0  5951.8     .16       0
Bank Sta=4872.3,5149.3
XS Rating Curve= 0 ,0
Exp/Cntr=0.3,0.1

Type RM Length L Ch R = 1 ,39599   ,964,964,964
BEGIN DESCRIPTION:
Mapping XS 9affa583
END DESCRIPTION:
XS GIS Cut Line= 3
      2858667.56     10099613.27      2859586.98     10098025.17
      2859865.59     10096729.63
#Sta/Elev= 30
  2818.2 1443.61  2878.6 1440.96    2928 1438.03  3060.9 1427.93  3244.3 1409.37
  3491.1 1371.63  3768.4 1359.41  3819.2 1357.95  3894.9 1355.97  4204.6 1350.79
  4545.8 1335.15  4716.1 1323.13    4757 1316.83  4796.1 1310.11  4825.1 1303.01
  4910.4    1306  4989.3  1302.1    4992  1301.6  4995.3  1302.1  5017.4  1302.6
  5053.6 1318.07  5073.3 1322.58  5196.8 1333.31  5416.6 1342.61  5584.6  1351.1
  5657.1 1353.89  5682.8 1361.25  5749.2 1366.84    5831 1383.88  5978.4 1398.29
#Mann= 14 ,-1 , 0
  2818.2      .1       0  2878.6     .16       0    2928      .1       0
  3060.9     .16       0  3768.4      .1       0  3819.2     .16       0
  3894.9      .1       0  4204.6     .16       0  4796.1      .1       0
  4989.3     .07       0  4995.3      .1       0  5073.3     .16       0
  5416.6      .1       0  5584.6     .16       0
Bank Sta=4757,5053.6
XS Rating Curve= 0 ,0
Exp/Cntr=0.3,0.1

Type RM Length L Ch R = 1 ,38635   ,1133,1133,1133
BEGIN DESCRIPTION:
NORTH GRAPE CREEK 46.0
END DESCRIPTION:
XS GIS Cut Line= 3
      2860938.25      10100226.2      2860436.75     10098443.09
      2860478.54     10097189.38
#Sta/Elev= 30
  2722.1 1414.44  2891.8 1408.71  2959.9 1403.13  3046.7 1399.63  3119.4 1393.39
  3365.6 1381.96  3737.3 1369.33  3810.6 1364.48  3923.1 1361.38  4216.3 1346.92
  4613.8 1335.09  4763.9 1323.81  4833.9 1311.88  4883.9 1302.84  4920.9 1299.93
  4923.7 1299.43  4926.9 1299.93  4960.2 1302.09  5077.5 1301.65  5114.1 1304.23
  5149.9 1311.96  5154.1 1312.97  5194.1 1319.62  5484.3 1332.83  5554.3 1337.88
  5573.9  1341.4  5614.3 1349.33  5654.4 1361.64  5710.3 1365.07  5828.8 1365.19
#Mann= 7 ,-1 , 0
  2722.1     .16       0  4920.9     .07       0  4926.9     .16       0
  4960.2      .1       0  5149.9     .16       0  5573.9      .1       0
  5710.3     .16       0
Bank Sta=4833.9,5154.1
XS Rating Curve= 0 ,0
Exp/Cntr=0.3,0.1

Type RM Length L Ch R = 1 ,37502   ,1012,1012,1012
BEGIN DESCRIPTION:
NORTH GRAPE CREEK 45.0
END DESCRIPTION:
XS GIS Cut Line= 3
        2861593.     10099989.36      2861495.48     10097593.32
        2861189.     10096673.88
#Sta/Elev= 30
  2995.2 1411.36  3350.3 1388.25  3475.8 1381.97  3718.9 1364.93  3871.6 1360.32
  4201.8  1344.2  4502.1 1334.04  4592.2 1325.46  4772.3  1319.1  4892.4 1312.52
  4942.4 1306.72  4962.2 1295.69  4982.5 1289.91  4999.5  1289.5  5002.2    1289
  5005.5  1289.5  5082.6 1296.83  5172.6  1300.3  5191.2 1303.42  5202.7 1305.11
  5366.9  1308.9  5441.4 1311.79  5474.4 1313.61  5525.3 1318.76  5606.3 1322.38
    5752 1330.64  5867.1 1344.78  6025.2 1349.42  6151.7 1361.03  6362.4 1374.28
#Mann= 10 ,-1 , 0
  2995.2      .1       0  3350.3     .16       0  4962.2      .1       0
  4999.5     .07       0  5005.5      .1       0  5191.2     .16       0
  5366.9      .1       0  5441.4     .16       0  5474.4     .05       0
  5606.3     .16       0
Bank Sta=4942.4,5202.7
XS Rating Curve= 0 ,0
Exp/Cntr=0.3,0.1

Type RM Length L Ch R = 1 ,36490   ,1239,1239,1239
BEGIN DESCRIPTION:
NORTH GRAPE CREEK 44.0
END DESCRIPTION:
XS GIS Cut Line= 3
      2862484.56     10098624.17      2862470.63     10097885.86
      2862331.32     10096743.57
#Sta/Elev= 30
  4059.7 1390.08  4078.3 1388.42  4121.4 1385.88  4370.2 1352.94  4510.2 1338.97
  4646.5 1320.56  4651.5 1323.77  4790.3 1316.27  4856.5 1307.28  4861.5 1308.93
  4880.9 1302.88  4921.2 1291.58  4951.4 1287.38  4988.7 1285.67  4991.4 1285.17
  4994.7 1285.67    5032 1286.45  5062.2 1292.01  5106.3 1292.85    5163    1302
  5164.1 1301.95  5193.2 1301.92  5223.4 1307.83  5437.8  1324.1  5495.4 1330.66
  5616.3 1353.16  5777.5 1365.25  5845.8 1375.01  5850.8 1371.79  5948.9 1387.33
#Mann= 6 ,-1 , 0
  4059.7      .1       0  4078.3     .16       0  4951.4      .1       0
  4988.7     .07       0  4994.7      .1       0  5164.1     .16       0
Bank Sta=4880.9,5163
XS Rating Curve= 0 ,0
Exp/Cntr=0.3,0.1

Type RM Length L Ch R = 1 ,35251   ,935,935,935
BEGIN DESCRIPTION:
NORTH GRAPE CREEK 41.0
END DESCRIPTION:
XS GIS Cut Line= 3
      2863041.76     10098986.42      2863654.73     10097983.38
      2863766.08     10096577.59
#Sta/Elev= 30
  3490.2 1362.35  3574.9 1355.93  3603.8  1354.4  3788.6  1342.4  3857.1 1338.43
  3972.4 1333.86  3984.5  1333.3    4194 1324.08  4664.5 1304.04  4778.5 1302.18
  4900.4 1291.98    4907 1291.97  4926.2 1287.17  4993.4 1282.71  4996.1 1282.21
  4999.4 1282.71  5046.5 1283.74  5106.7 1290.11    5177 1291.66  5237.1 1297.27
  5277.3 1294.26  5307.4 1295.72  5367.5 1303.65  5467.9 1311.42  5530.8 1322.06
  5548.1 1325.78  5618.3 1333.52    5839 1349.18  6043.7 1372.07  6075.9 1377.87
#Mann= 12 ,-1 , 0
  3490.2     .16       0  3574.9     .05       0  3603.8     .16       0
  3788.6     .05       0  3857.1      .1       0  3972.4     .05       0
  3984.5      .1       0    4194     .05       0  4900.4      .1       0
  4993.4     .07       0  4999.4      .1       0  5530.8     .16       0
Bank Sta=4907,5106.7
XS Rating Curve= 0 ,0
Exp/Cntr=0.3,0.1

Type RM Length L Ch R = 1 ,34316   ,1486,1486,1486
BEGIN DESCRIPTION:
NORTH GRAPE CREEK 40.0
END DESCRIPTION:
XS GIS Cut Line= 3
      2864225.89     10099613.29      2864629.88     10097300.78
      2864504.51     10096673.93
#Sta/Elev= 30
  3162.9 1320.07  3431.7 1312.78  3477.1 1309.39  3571.8 1312.77  3662.1 1311.54
  3793.8 1310.37  3861.4 1309.82  4102.7  1307.4  4269.1  1306.3  4460.6  1305.6
  4652.7 1299.41  4952.2 1291.86  4958.9 1289.69  4986.7 1282.93  4989.5 1282.43
  4992.7 1282.93    5058 1283.61  5101.4 1284.12  5131.8 1289.87  5157.1 1290.42
  5247.4 1290.22  5325.9 1293.15  5375.5 1305.16    5413 1310.83  5578.8 1326.66
  5854.2 1346.33  5894.9 1352.56    5951 1366.45    6002 1373.72  6149.7 1385.52
#Mann= 17 ,-1 , 0
  3162.9      .1       0  3431.7     .16       0  3571.8      .1       0
  3662.1     .05       0  3793.8      .1       0  3861.4     .05       0
  4102.7      .1       0  4269.1     .05       0  4460.6      .1       0
  4652.7     .05       0  4958.9      .1       0  4986.7     .07       0
  4992.7      .1       0    5058     .05       0  5157.1     .16       0
  5247.4     .05       0  5325.9     .16       0
Bank Sta=4952.2,5131.8
XS Rating Curve= 0 ,0
Exp/Cntr=0.3,0.1

Type RM Length L Ch R = 1 ,32830   ,786,786,786
BEGIN DESCRIPTION:
NORTH GRAPE CREEK 38.0
END DESCRIPTION:
XS GIS Cut Line= 3
      2865382.13     10099195.34      2865827.91     10097481.88
      2865772.42     10097107.27
#Sta/Elev= 30
  3553.1 1329.83  3828.2 1320.39  3863.8 1319.14  4018.5 1311.19  4380.8 1295.43
  4511.1 1289.58  4567.4 1289.02  4701.7 1285.95  4749.1 1282.16  4819.8 1283.89
  4970.4  1281.7  4989.2 1277.96    4992 1277.46  4995.2 1277.96  5068.1 1279.96
  5094.4 1284.79  5097.9 1285.31  5184.5 1297.83  5230.2 1302.15  5265.5 1312.01
  5271.3 1311.71  5298.9 1319.98  5306.1 1319.95  5320.1 1327.94  5350.5    1339
  5432.9 1360.22  5494.5  1368.7  5544.1 1372.68  5574.5 1377.95  5702.3 1391.45
#Mann= 12 ,-1 , 0
  3553.1      .1       0  3828.2     .16       0  3863.8      .1       0
  4018.5     .16       0  4380.8      .1       0  4567.4     .16       0
  4819.8      .1       0  4989.2     .07       0  4995.2      .1       0
  5097.9     .16       0  5271.3     .05       0  5298.9     .16       0
Bank Sta=4970.4,5094.4
XS Rating Curve= 0 ,0
Exp/Cntr=0.3,0.1

Type RM Length L Ch R = 1 ,32044   ,759,759,759
BEGIN DESCRIPTION:
NORTH GRAPE CREEK 37.0
END DESCRIPTION:
XS GIS Cut Line= 3
      2865730.39     10099167.51      2866608.03     10097788.35
      2866844.85     10096924.66
#Sta/Elev= 30
  3597.4 1326.89  3696.8 1323.97  3734.2 1323.51  3981.4 1319.16    4127 1310.41
    4193 1310.37  4272.6 1308.07    4403 1295.58  4464.5 1294.37  4763.7 1276.72
  4830.6 1281.23  4903.4 1280.82  4967.7 1273.42  5000.3 1273.04    5003 1272.54
  5006.3 1273.04  5039.7 1274.26  5054.9 1278.25  5127.7  1292.9    5253  1299.6
    5548 1320.73  5693.2 1328.13  5755.4 1337.59  5789.6  1347.4  5879.8 1376.09
  5935.1 1384.25  5969.6 1395.68  5974.8 1394.33  6043.7 1405.17  6127.7 1411.48
#Mann= 10 ,-1 , 0
  3597.4      .1       0  3696.8     .16       0  3734.2      .1       0
    4193     .16       0  4464.5      .1       0  4967.7     .16       0
  5000.3     .07       0  5006.3     .16       0    5253      .1       0
  5789.6     .16       0
Bank Sta=4903.4,5054.9
XS Rating Curve= 0 ,0
Exp/Cntr=0.3,0.1

Type RM Length L Ch R = 1 ,31285   ,597,597,597
BEGIN DESCRIPTION:
NORTH GRAPE CREEK 36.0
END DESCRIPTION:
XS GIS Cut Line= 3
      2866440.87     10099780.41      2867290.63     10097941.59
      2867694.03     10097134.79
#Sta/Elev= 30
  3313.5 1354.47  3384.2 1352.38  3672.6 1338.01  3775.3  1328.6  3838.6 1330.03
  3987.2 1320.09    4093 1321.17  4199.2 1317.36  4324.9 1302.73  4573.6 1287.55
    4634 1283.24  4682.3 1274.72  4885.2 1276.27  4907.2 1272.23  5014.5 1269.36
  5017.3 1268.86  5020.5 1269.36  5053.2 1275.25  5063.4 1276.68  5132.2 1280.09
  5171.6  1295.1    5201 1298.87  5359.4 1301.11  5522.8 1306.24  5658.3 1319.74
  5715.4 1323.21  5851.1 1330.26  5992.7 1344.72  6126.6 1364.58  6241.2 1373.82
#Mann= 12 ,-1 , 0
  3313.5      .1       0  3384.2     .16       0    4093      .1       0
  4573.6     .16       0  4682.3      .1       0  5014.5     .07       0
  5020.5      .1       0  5053.2     .16       0  5359.4      .1       0
  5658.3     .16       0  5715.4      .1       0  5992.7     .16       0
Bank Sta=4885.2,5063.4
XS Rating Curve= 0 ,0
Exp/Cntr=0.3,0.1

Type RM Length L Ch R = 1 ,30688   ,963,963,963
BEGIN DESCRIPTION:
Mapping XS 97c8f163
END DESCRIPTION:
XS GIS Cut Line= 3
       2868523.2     10099857.75      2867741.98     10099154.65
      2867676.87     10097318.73
#Sta/Elev= 30
  3184.9 1324.96  3299.7 1321.32  3371.1 1317.69  3495.7 1307.37  3580.9 1306.61
  3622.7  1311.1  3741.7 1299.19    3917 1290.11  4010.2 1286.36  4071.3 1284.73
  4138.1 1281.92  4379.2 1280.03  4572.9 1266.67  4657.1 1263.49  4717.1 1277.21
  4835.7 1276.78  4897.3 1275.66  4927.3 1268.34  4994.3 1263.11  4997.1 1262.61
  5000.3 1263.11  5052.4 1274.53  5067.4 1276.67  5217.5 1276.65  5357.5 1302.17
    5472 1308.78  5737.8 1329.45  5817.8 1326.21  5988.9 1347.17    6073 1358.14
#Mann= 16 ,-1 , 0
  3184.9      .1       0  3299.7     .05       0  3371.1      .1       0
  3741.7     .05       0    3917     .16       0  4010.2      .1       0
  4071.3     .16       0  4138.1      .1       0  4379.2     .05       0
  4572.9     .16       0  4835.7      .1       0  4994.3     .07       0
  5000.3      .1       0  5052.4     .16       0    5472      .1       0
  5988.9     .16       0
#XS Ineff= 2 , 0
         4236.78 1282.94
Permanent Ineff=
       F       F
Bank Sta=4897.3,5067.4
XS Rating Curve= 0 ,0
Exp/Cntr=0.3,0.1

Type RM Length L Ch R = 1 ,29725   ,834,834,834
BEGIN DESCRIPTION:
NORTH GRAPE CREEK 34.0
END DESCRIPTION:
XS GIS Cut Line= 2
      2869143.41     10099042.11      2867708.56     10097189.34
#Sta/Elev= 30
    4030  1399.5  4219.2 1398.59  4488.4 1388.72  4573.5 1383.14  4623.3 1375.36
  4716.6 1349.03  4766.4 1328.02  4780.8 1316.66  4830.6  1296.1  4845.1 1285.31
  4874.1 1276.09  4915.7 1268.86  4951.3 1257.54  4985.6 1257.72  5026.8 1257.31
  5029.6 1256.81  5032.8 1257.31  5137.6 1269.27  5187.4 1269.57  5243.5 1276.19
  5485.5 1289.71  5602.1 1294.93    5679 1301.39  5728.8 1312.56  5817.8 1318.31
  5913.5 1329.24  6021.2 1334.34  6120.8 1349.05  6255.7 1362.86  6373.4 1368.72
#Mann= 8 ,-1 , 0
    4030     .05       0  4219.2     .16       0  4985.6      .1       0
  5026.8     .07       0  5032.8      .1       0  5485.5     .05       0
  5602.1      .1       0  5817.8     .16       0
Bank Sta=4915.7,5137.6
XS Rating Curve= 0 ,0
Exp/Cntr=0.3,0.1

Type RM Length L Ch R = 1 ,28891   ,1471,1471,1471
BEGIN DESCRIPTION:
NORTH GRAPE CREEK 33.0
END DESCRIPTION:
XS GIS Cut Line= 3
      2870968.35     10098777.44      2868934.45      10097676.9
       2868098.6     10096868.91
#Sta/Elev= 30
  3015.2 1359.17  3208.5 1351.59  3318.2  1347.6  3356.5 1345.24  3587.2 1329.18
  3704.4 1333.06  3855.5 1324.15  3866.5 1322.66  3976.1 1312.06  4065.6 1302.98
  4095.2 1297.78  4256.2 1299.43  4368.1 1292.14  4441.7 1297.83  4545.4 1286.29
    4611  1288.6  4692.8 1276.59    4884 1271.74  4908.9 1266.85    4944 1259.28
  5058.7 1255.97  5061.4 1255.47  5064.7 1255.97  5199.1 1267.54    5217 1269.75
    5365    1276  6034.3 1304.45  6310.1 1337.56  6421.2  1345.9  6490.3 1350.65
#Mann= 15 ,-1 , 0
  3015.2     .05       0  3208.5     .16       0  3318.2      .1       0
  3356.5     .16       0  3587.2     .05       0  3855.5     .16       0
  3866.5     .05       0  3976.1      .1       0  4065.6     .16       0
  4908.9      .1       0  5058.7     .07       0  5064.7      .1       0
  5199.1     .16       0    5365     .05       0  6421.2      .1       0
#XS Ineff= 2 , 0
         4593.22 1289.38
Permanent Ineff=
       F       F
Bank Sta=4884,5217
XS Rating Curve= 0 ,0
Exp/Cntr=0.3,0.1

Type RM Length L Ch R = 1 ,27420   ,755,755,755
BEGIN DESCRIPTION:
NORTH GRAPE CREEK 30.0
END DESCRIPTION:
XS GIS Cut Line= 2
       2869519.5     10096464.94       2867945.4     10096687.82
#Sta/Elev= 30
  4419.9  1371.4  4446.6 1367.07  4481.5 1369.19  4542.1 1367.12    4628 1353.74
  4774.4 1330.77  4801.6 1324.79  4843.2 1310.53  4872.6 1291.36  4877.7 1290.58
  4905.7 1265.68  4925.9 1258.09  4983.5 1253.69  4986.3 1253.19  4989.5 1253.69
  5077.4 1255.51    5138 1254.03  5185.6 1258.25  5190.2 1258.32  5227.7 1261.94
  5303.8 1271.77  5390.5 1295.24  5531.9 1304.43  5601.1    1314  5630.9 1316.21
  5663.9 1323.18  5731.1 1326.02  5831.4 1332.72  5871.9 1340.42  6009.7 1355.09
#Mann= 11 ,-1 , 0
  4419.9      .1       0    4628     .16       0  4843.2      .1       0
  4983.5     .07       0  4989.5      .1       0  5185.6     .05       0
  5190.2      .1       0  5601.1     .16       0  5630.9      .1       0
  5731.1     .16       0  5831.4      .1       0
Bank Sta=4905.7,5227.7
XS Rating Curve= 0 ,0
Exp/Cntr=0.3,0.1

Type RM Length L Ch R = 1 ,26665   ,987,987,987
BEGIN DESCRIPTION:
Mapping XS 82aa873b
END DESCRIPTION:
XS GIS Cut Line= 3
      2869282.75     10095907.71      2868391.15      10095991.3
      2867666.79     10096395.27
#Sta/Elev= 30
  4350.4 1298.83  4404.9 1296.16    4424  1297.4  4469.4 1301.52  4535.5 1296.36
  4692.2 1274.25  4791.7 1263.17  4826.8  1258.8  4856.9 1253.55    4884 1251.91
  4886.8 1251.41    4890 1251.91  4891.2 1251.92  4897.7 1252.12  4990.7 1252.61
  5047.7  1255.9  5128.1 1253.62  5188.3 1258.82  5238.6 1260.85  5301.4 1273.26
  5382.5  1284.2  5500.9 1295.26  5550.5 1306.55  5588.2 1321.54  5788.6 1343.23
  5815.6 1347.67  5875.2 1351.89  5905.7 1353.65    5991 1358.49  6075.3 1364.27
#Mann= 13 ,-1 , 0
  4350.4     .05       0    4424      .1       0  4692.2     .16       0
  4791.7     .05       0    4884     .07       0    4890     .05       0
  4891.2     .16       0  4897.7     .05       0  4990.7      .1       0
  5788.6     .16       0  5875.2      .1       0  5905.7     .16       0
    5991     .05       0
Bank Sta=4826.8,5188.3
XS Rating Curve= 0 ,0
Exp/Cntr=0.3,0.1

Type RM Length L Ch R = 1 ,25678   ,1075,1075,1075
BEGIN DESCRIPTION:
NORTH GRAPE CREEK 28.0
END DESCRIPTION:
XS GIS Cut Line= 3
      2869018.06     10095155.45      2867917.51     10095517.65
       2867499.6     10096214.18
#Sta/Elev= 30
  4308.1 1290.21  4416.4  1288.5  4470.2 1288.53  4541.2 1285.65  4644.6 1267.74
  4781.4 1256.34  4855.1 1254.75  4907.8 1248.59  4999.5  1245.8  5002.2  1245.3
  5005.5  1245.8  5034.1  1246.4  5057.4 1250.93  5082.3 1252.05  5097.2 1254.69
  5202.5 1260.32  5301.3 1271.85  5406.7 1274.09  5481.2 1278.97  5555.7 1284.94
    5593  1287.6  5762.3 1299.87  5816.6 1304.05  5980.5 1319.94  6017.4  1330.9
  6038.8  1334.7  6075.8 1346.83  6112.7 1352.48  6263.9 1362.12    6279 1362.71
#Mann= 15 ,-1 , 0
  4308.1     .05       0  4416.4      .1       0  4470.2     .05       0
  4541.2      .1       0  4999.5     .07       0  5005.5      .1       0
  5082.3     .05       0  5301.3      .1       0  5406.7     .05       0
  5481.2      .1       0  5555.7     .16       0    5593      .1       0
  5762.3     .05       0  5816.6      .1       0  6263.9     .05       0
Bank Sta=4855.1,5097.2
XS Rating Curve= 0 ,0
Exp/Cntr=0.3,0.1

Type RM Length L Ch R = 1 ,24603   ,855,855,855
BEGIN DESCRIPTION:
NORTH GRAPE CREEK 26.0
END DESCRIPTION:
XS GIS Cut Line= 3
      2868781.22     10094389.27      2866844.85     10094528.58
       2866288.4     10095029.38
#Sta/Elev= 30
  4172.2 1272.15  4320.2 1272.84  4385.5  1272.1  4581.9 1260.99  4726.8 1255.75
  4776.5 1248.62  4816.6 1251.86  4846.7 1244.55  4886.8 1246.71  4935.6 1245.28
    4967 1244.02  4993.5    1240  4996.2  1239.5  4999.5    1240  5034.8 1246.08
  5134.1 1253.33  5147.5 1255.14  5267.8 1255.81  5431.8 1260.53  5678.8 1263.42
    5826 1271.31  5874.2 1273.45  6027.3 1278.67  6131.6 1279.96  6214.8 1282.35
  6269.7 1285.08  6407.8 1286.51  6426.3  1285.7  6460.3 1288.65  6862.2 1306.19
#Mann= 16 ,-1 , 0
  4172.2     .05       0  4320.2      .1       0  4935.6     .05       0
  4993.5    .035       0  4999.5     .05       0  5034.8      .1       0
  5134.1     .16       0  5431.8     .05       0    5826      .1       0
  5874.2     .05       0  6027.3     .16       0  6131.6     .05       0
  6214.8      .1       0  6269.7     .05       0  6407.8      .1       0
  6460.3     .05       0
#XS Ineff= 2 , 0
         4277.85  1272.8
Permanent Ineff=
       F       F
Bank Sta=4726.8,5147.5
XS Rating Curve= 0 ,0
Exp/Cntr=0.3,0.1

Type RM Length L Ch R = 1 ,23748   ,939,939,939
BEGIN DESCRIPTION:
NORTH GRAPE CREEK 25.0
END DESCRIPTION:
XS GIS Cut Line= 2
      2868962.29     10094208.16      2866413.26     10092592.38
#Sta/Elev= 30
  3919.8 1272.27  4121.9 1273.52  4272.7 1270.62  4539.4 1257.07    4571 1247.57
  4592.2 1245.65  4639.5 1251.92  4765.1 1252.24  4816.8 1249.68  4837.9 1244.25
    4957 1238.87  4980.7 1237.19  4983.4 1236.69  4986.7 1237.19  5035.4 1238.22
  5084.6 1250.81  5171.8 1251.04  5208.2 1255.57  5259.9 1256.82    5287 1263.14
  5326.2 1263.51  5375.2 1273.58  5425.5 1273.01  5636.2 1269.78  5803.1 1274.09
  6027.6  1285.4  6302.9  1289.8  6765.3 1318.22  6831.8 1318.28  6937.8 1312.51
#Mann= 11 ,-1 , 0
  3919.8     .05       0  4272.7      .1       0  4539.4     .05       0
  4639.5      .1       0    4957     .16       0  4980.7     .07       0
  4986.7     .16       0  5326.2      .1       0  5425.5     .05       0
  6302.9      .1       0  6765.3     .16       0
#XS Ineff= 2 , 0
         4108.05 1273.77 5387.71         1273.64
Permanent Ineff=
       F       F
Bank Sta=4816.8,5084.6
XS Rating Curve= 0 ,0
Exp/Cntr=0.3,0.1

Type RM Length L Ch R = 1 ,22809   ,771,771,771
BEGIN DESCRIPTION:
NORTH GRAPE CREEK 35.0
END DESCRIPTION:
XS GIS Cut Line= 3
      2868934.88     10094162.13      2868878.73     10093706.67
      2868892.66     10092243.94
#Sta/Elev= 30
  4364.8    1273  4554.6 1270.41  4716.4 1259.72  4806.5 1255.63  4809.2 1255.28
  4926.6 1233.99  4957.1  1232.8  4993.7 1232.34  4996.4 1231.84  4999.7 1232.34
  5036.7 1235.54  5046.7  1235.7  5076.7 1243.27  5106.7 1255.93  5126.7 1260.01
  5156.7 1259.79  5220.4  1273.9  5256.7 1277.94  5316.5 1275.12  5366.7 1276.92
  5426.7 1283.76  5506.7 1278.07  5546.7 1279.94  5596.7 1276.97  5671.5 1283.74
  5756.7 1291.59  5816.7 1293.26    5997 1288.64  6103.9 1286.75  6286.5 1285.45
#Mann= 11 ,-1 , 0
  4364.8     .05       0  4716.4      .1       0  4809.2     .05       0
  4957.1      .1       0  4993.7     .07       0  4999.7      .1       0
  5036.7     .16       0  5220.4      .1       0  5671.5     .16       0
    5997      .1       0  6103.9     .05       0
Bank Sta=4806.5,5106.7
XS Rating Curve= 0 ,0
Exp/Cntr=0.3,0.1

Type RM Length L Ch R = 1 ,22038   ,1116,1116,1116
BEGIN DESCRIPTION:
NORTH GRAPE CREEK 24.0
END DESCRIPTION:
XS GIS Cut Line= 3
      2869268.78     10094960.45       2869728.5      10093358.4
      2869436.28     10092467.82
#Sta/Elev= 30
  3764.1  1284.1  3851.5 1280.29  4287.4  1263.2  4471.6 1260.42    4578 1256.69
  4780.2 1253.92  4789.2 1253.38    4796 1251.45  4801.2 1252.12  4863.5 1243.26
  4894.7 1242.83  4938.1 1237.63  4957.1  1230.8  4995.7 1230.05  4998.5 1229.55
  5001.7 1230.05  5040.3 1230.91  5061.1 1240.16  5071.5 1242.02  5159.4 1249.85
  5193.1 1254.77  5382.2 1257.78  5389.1 1258.01  5507.1  1261.6  5698.6 1263.99
  5767.5 1267.16  5825.1 1267.57  5881.4 1270.68  6015.8    1278  6368.1 1290.13
#Mann= 11 ,-1 , 0
  3764.1      .1       0  3851.5     .05       0  4789.2      .1       0
  4938.1     .16       0  4995.7     .07       0  5001.7     .16       0
  5382.2      .1       0  5389.1     .16       0  5507.1      .1       0
  5881.4     .16       0  6015.8      .1       0
Bank Sta=4780.2,5193.1
XS Rating Curve= 0 ,0
Exp/Cntr=0.3,0.1

Type RM Length L Ch R = 1 ,20922   ,1178,1178,1178
BEGIN DESCRIPTION:
NORTH GRAPE CREEK 23.0
END DESCRIPTION:
XS GIS Cut Line= 3
      2870313.59     10095169.35       2870773.3     10093637.02
      2870801.16     10092912.66
#Sta/Elev= 30
  3878.5  1281.9  4054.3 1277.72  4167.4 1267.86  4367.6 1255.62  4456.1 1253.68
  4474.2  1253.4  4675.5 1254.24  4889.6 1249.58  4907.5 1247.86  4959.3 1235.45
    4991 1229.92  4993.7 1229.42    4997 1229.92  5105.9 1231.29  5126.2 1240.25
  5154.2 1245.23  5202.8 1249.64    5252 1251.87  5325.1 1252.61    5428 1257.79
  5550.3 1265.95  5581.7 1268.12  5641.7 1267.61  5681.7 1272.17  5724.3 1274.39
  5871.9 1281.19  5931.9 1281.78  6005.1  1285.1    6072 1285.06  6203.2 1281.82
#Mann= 11 ,-1 , 0
  3878.5      .1       0  4167.4     .05       0  4456.1      .1       0
  4474.2     .05       0  4959.3      .1       0    4991     .07       0
    4997      .1       0  5154.2     .16       0    5428      .1       0
  5550.3     .05       0  5724.3      .1       0
#XS Ineff= 2 , 0
         4661.63 1254.38
Permanent Ineff=
       F       F
Bank Sta=4889.6,5202.8
XS Rating Curve= 0 ,0
Exp/Cntr=0.3,0.1
