HEC-RAS study PALO ALTO CREEK.prj: PALO ALTO CREEK Base Level Engineering

--- PALO ALTO CREEK.g01 (geometry) --- (continued)

Type RM Length L Ch R = 1 ,38712   ,1113,1113,1113
BEGIN DESCRIPTION:
Mapping XS 89d2525c
END DESCRIPTION:
XS GIS Cut Line= 3
      2776022.62      10078185.1      2775633.73     10077032.34
      2774515.66     10076185.11
#Sta/Elev= 30
  3619.3 1653.65  3741.9 1651.03  3864.3 1645.12    3957 1639.61  4000.7 1635.28
  4032.3 1633.47  4082.9 1631.77  4122.3 1632.89  4543.6 1633.78    4839 1635.41
  4853.6 1634.37  4909.8  1626.4  5000.4 1614.66  5003.1 1614.16  5006.4 1614.66
  5030.7 1619.95  5059.6 1622.61  5088.7 1627.43  5138.6 1633.71  5153.2  1634.6
  5209.4 1634.42  5323.8 1636.43  5417.4 1639.58  5488.1 1639.09  5502.7 1640.95
  5552.6 1642.61  5573.4 1641.78  5761.6 1644.37  6166.3 1652.76  6238.7 1652.98
#Mann= 7 ,-1 , 0
  3619.3     .05       0  3864.3      .1       0  4122.3     .05       0
  4543.6      .1       0  5000.4     .07       0  5006.4      .1       0
  5761.6     .05       0
#XS Ineff= 2 , 0
         4838.57 1635.45
Permanent Ineff=
       F       F
Bank Sta=4909.8,5088.7
XS Rating Curve= 0 ,0
Exp/Cntr=0.3,0.1

Type RM Length L Ch R = 1 ,37599   ,955,955,955
BEGIN DESCRIPTION:
PALO ALTO CREEK 56.0
END DESCRIPTION:
XS GIS Cut Line= 3
      2776182.35     10078101.81      2776057.35     10076129.57
      2775689.29     10075032.35
#Sta/Elev= 30
  2865.3 1651.13  2943.5  1650.3  3077.8 1644.86  3094.1 1643.95  3113.9  1641.5
    3174 1642.25  3227.5 1640.73  3264.2 1635.83  3424.5 1628.88  3544.7  1631.1
  3621.7 1630.85  4587.7 1631.09  4626.9 1631.32  4807.3 1622.36    4932 1615.75
  4962.3 1615.95  4992.3 1613.55  4995.1 1613.05  4998.3 1613.55  5016.4 1614.33
  5042.6 1620.58  5068.8 1621.79  5142.4    1630  5163.5 1632.66  5248.5 1636.88
  5429.3 1640.38  5486.5 1640.97  5836.6 1647.54  5968.9 1651.38  5998.8 1652.38
#Mann= 14 ,-1 , 0
  2865.3     .05       0  3077.8      .1       0  3094.1     .05       0
  3227.5      .1       0  3621.7     .05       0  4587.7      .1       0
  4962.3     .16       0  4992.3     .07       0  4998.3     .16       0
  5142.4      .1       0  5429.3     .16       0  5486.5      .1       0
  5836.6     .05       0  5968.9      .1       0
#XS Ineff= 2 , 0
         3553.81 1631.19
Permanent Ineff=
       F       F
Bank Sta=4807.3,5042.6
XS Rating Curve= 0 ,0
Exp/Cntr=0.3,0.1

Type RM Length L Ch R = 1 ,36644   ,750,750,750
BEGIN DESCRIPTION:
PALO ALTO CREEK 55.0
END DESCRIPTION:
XS GIS Cut Line= 3
       2776376.8     10078011.47      2776571.23     10076678.18
      2776960.14     10075962.86
#Sta/Elev= 30
  3522.3 1647.69  3606.7 1648.33  3701.9 1646.92  3833.3 1641.67    3903  1635.9
    3977 1632.71  4227.4 1625.89  4409.3 1629.01  4865.1 1628.13  4915.4  1624.3
  4975.3 1616.33  4988.6 1608.06  4999.8 1606.98  5002.6 1606.48  5005.8 1606.98
    5019 1608.83  5034.1 1607.64  5056.9 1611.59  5062.7 1613.83    5091 1614.11
  5128.2 1612.45  5150.1 1615.69  5197.9 1618.61  5226.1 1620.02  5335.3 1633.73
    5387 1637.66  5480.3 1641.62    5647 1645.02  5658.5 1644.95  5683.9 1644.41
#Mann= 11 ,-1 , 0
  3522.3      .1       0  3606.7     .05       0    3903      .1       0
    3977     .05       0  4865.1      .1       0  4999.8     .07       0
  5005.8      .1       0  5197.9     .16       0  5480.3     .05       0
    5647      .1       0  5658.5     .05       0
#XS Ineff= 2 , 0
         4414.78 1628.97
Permanent Ineff=
       F       F
Bank Sta=4975.3,5062.7
XS Rating Curve= 0 ,0
Exp/Cntr=0.3,0.1

Type RM Length L Ch R = 1 ,35894   ,561,561,561
BEGIN DESCRIPTION:
PALO ALTO CREEK 53.0
END DESCRIPTION:
XS GIS Cut Line= 4
      2777161.51     10077657.39      2777251.79     10076969.84
      2777369.85     10076699.01      2777244.85     10076358.74
#Sta/Elev= 30
  4237.2 1633.56  4301.4 1633.89  4403.9 1628.99    4559 1625.59  4704.8 1625.54
  4716.5 1623.99  4765.4 1622.14  4791.4 1619.89    4869 1613.27  4906.6 1612.05
  4930.7 1609.58  4933.4 1608.25  4948.2  1606.3  4962.2 1605.26  4980.2 1605.96
  5011.5  1603.1  5014.3  1602.6  5017.5  1603.1  5024.6  1606.9  5032.5 1612.89
  5055.9 1616.15  5084.8 1623.07  5108.2 1626.13    5218 1626.45  5351.7 1627.27
  5446.8    1629  5519.4 1631.97  5540.7 1635.48  5553.2 1635.94  5588.6 1635.76
#Mann= 9 ,-1 , 0
  4237.2      .1       0  4403.9     .05       0  4791.4      .1       0
  5011.5     .07       0  5017.5      .1       0    5218     .05       0
  5351.7      .1       0  5446.8     .05       0  5553.2      .1       0
Bank Sta=4906.6,5032.5
XS Rating Curve= 0 ,0
Exp/Cntr=0.3,0.1

Type RM Length L Ch R = 1 ,35333   ,839,839,839
BEGIN DESCRIPTION:
PALO ALTO CREEK 52.0
END DESCRIPTION:
XS GIS Cut Line= 4
      2777407.38     10077711.44      2777778.94     10077357.24
      2777633.11     10076541.27      2777285.89     10076124.61
#Sta/Elev= 30
  4319.4 1630.29  4367.2  1628.4  4465.8 1625.74    4637 1623.48  4887.1 1622.61
  4921.7 1619.43  4937.9 1620.62    4948 1619.91  4958.2 1613.47  4968.4 1606.71
  4975.5 1603.33  4998.6 1600.86  5034.4    1603  5049.6 1605.82  5059.8 1606.04
  5080.1 1604.58  5088.2  1605.2  5110.6 1609.37    5141 1612.03  5215.7 1617.42
  5262.7  1618.8  5293.4 1619.56  5372.5 1623.61  5452.4 1624.05  5761.7 1625.06
  5813.9 1625.49    5883 1627.35  5968.9 1632.25  6160.3 1640.78    6204 1641.36
#Mann= 10 ,-1 , 0
  4319.4     .05       0  4367.2      .1       0  4465.8     .05       0
  4958.2    .035       0    5141      .1       0  5215.7     .05       0
  5262.7      .1       0  5452.4     .05       0  5761.7      .1       0
  5813.9     .05       0
Bank Sta=4958.2,5141
XS Rating Curve= 0 ,0
Exp/Cntr=0.3,0.1

Type RM Length L Ch R = 1 ,34494   ,370,370,370
BEGIN DESCRIPTION:
PALO ALTO CREEK 51.0
END DESCRIPTION:
XS GIS Cut Line= 4
      2778570.61     10078471.83      2778692.13     10077985.71
      2778313.66     10077176.68      2778362.27     10075860.74
#Sta/Elev= 30
  3094.3 1650.26  3307.9 1646.83  3395.6 1647.84  3608.6 1641.72  3665.9 1637.55
  3906.7 1620.47  3917.4  1617.9  3928.8 1610.39  3945.8    1604  4019.8 1598.25
  4065.5  1599.2  4082.8 1603.51  4193.7 1617.63  4278.2 1619.02  4571.6 1620.63
  4721.7 1619.52  4745.7 1617.37  4831.7 1609.49  4901.8 1607.88  5001.6  1596.6
  5025.9 1603.49  5031.9 1608.07  5041.9 1612.97  5061.9 1617.39    5162 1624.53
  5354.9 1628.51    5437 1628.46  5508.4 1629.41    5620  1631.7  5805.4 1634.81
#Mann= 10 ,-1 , 0
  3094.3     .05       0  3665.9      .1       0  4278.2     .05       0
  4745.7      .1       0  4901.8     .07       0  5031.9      .1       0
  5354.9     .05       0    5437      .1       0  5508.4     .05       0
    5620      .1       0
#XS Ineff= 2 , 0
         4515.81 1620.61
Permanent Ineff=
       F       F
Bank Sta=4901.8,5031.9
XS Rating Curve= 0 ,0
Exp/Cntr=0.3,0.1

Type RM Length L Ch R = 1 ,34124   ,557,557,557
BEGIN DESCRIPTION:
PALO ALTO CREEK 50.0
END DESCRIPTION:
XS GIS Cut Line= 3
      2778868.47     10077603.76      2778668.47     10076853.73
      2778468.46     10076403.71
#Sta/Elev= 30
  4186.6 1632.38  4279.1 1628.35  4324.4 1623.99  4352.2 1616.45  4372.9 1607.85
  4393.6 1604.99  4404.6 1599.07  4414.3 1596.72  4497.1 1598.86  4519.7 1605.28
  4528.2 1605.62  4559.9 1602.19  4589.6 1603.36    4642 1615.95  4662.7 1617.05
  4797.2 1613.37  4931.8 1604.55  4945.4 1604.12  4971.7    1597    4992 1595.81
  4994.7 1595.31    4998 1595.81  5029.2 1597.68    5047 1601.89  5052.4 1600.42
  5070.2 1606.45  5098.9 1608.38  5122.2 1613.59  5168.7 1618.14  5455.3 1623.86
#Mann= 3 ,-1 , 0
  4186.6      .1       0    4992     .07       0    4998      .1       0
#XS Ineff= 2 , 0
         4656.83 1617.06
Permanent Ineff=
       F       F
Bank Sta=4931.8,5070.2
XS Rating Curve= 0 ,0
Exp/Cntr=0.3,0.1

Type RM Length L Ch R = 1 ,33567   ,446,446,446
BEGIN DESCRIPTION:
PALO ALTO CREEK 49.0
END DESCRIPTION:
XS GIS Cut Line= 4
      2778773.84      10077926.1      2779131.89     10077370.59
      2779129.72     10076921.37      2778695.69     10076203.04
#Sta/Elev= 30
    4008 1642.61  4078.7 1640.93  4099.8 1638.63  4178.4 1635.09  4359.9 1631.45
  4411.4 1633.04  4468.8  1630.8  4505.1 1626.89  4526.2  1626.8  4556.6 1624.09
  4705.8 1619.85  4745.8 1616.02  4785.8 1608.54  4905.8 1603.16  4945.8 1597.53
  4982.8 1595.57  4985.5 1595.07  4988.8 1595.57  5035.8 1596.02  5057.2 1601.41
  5065.8  1604.3  5085.8 1611.14  5114.4  1615.3  5251.1 1615.59  5432.3 1618.19
  5547.7 1618.02    5576 1617.78  5656.3 1617.89  5781.3 1618.96  5957.4 1624.38
#Mann= 9 ,-1 , 0
    4008     .05       0  4982.8    .035       0  4988.8     .05       0
  5057.2      .1       0  5251.1     .05       0  5432.3      .1       0
  5547.7     .05       0    5576      .1       0  5656.3     .05       0
#XS Ineff= 2 , 0
                          5460.7         1618.72
Permanent Ineff=
       F       F
Bank Sta=4905.8,5065.8
XS Rating Curve= 0 ,0
Exp/Cntr=0.3,0.1

Type RM Length L Ch R = 1 ,33121   ,589,589,589
BEGIN DESCRIPTION:
PALO ALTO CREEK 48.0
END DESCRIPTION:
XS GIS Cut Line= 3
      2780220.14     10077495.48      2779393.72     10076766.29
       2778838.8     10075947.79
#Sta/Elev= 30
  4069.6 1643.19  4150.1 1633.49  4263.2 1623.11  4397.9  1616.2  4497.5 1613.98
  4688.2  1613.5  4879.8 1617.14    4894 1616.75  4914.9 1612.05  4936.7 1609.77
  4945.8 1606.78  4950.9 1605.61  4978.7 1595.07  4994.8  1592.7  4997.2 1592.69
    5000 1592.19  5003.2 1592.69  5049.6 1595.79  5067.7 1598.59  5134.9 1604.25
  5151.1 1604.76  5229.3 1609.33  5257.3 1611.96  5284.9 1616.92    5430 1616.76
  5522.8  1616.9  5775.5 1617.42  5940.2 1622.24  5961.2 1623.93  6160.6 1627.99
#Mann= 12 ,-1 , 0
  4069.6      .1       0  4150.1     .05       0  4945.8      .1       0
  4994.8     .05       0  4997.2    .035       0  5003.2     .05       0
  5067.7      .1       0  5151.1     .05       0  5229.3      .1       0
  5284.9     .05       0    5430      .1       0  5522.8     .05       0
#XS Ineff= 2 , 0
         4879.69 1616.91 5290.81         1616.91
Permanent Ineff=
       F       F
Bank Sta=4950.9,5134.9
XS Rating Curve= 0 ,0
Exp/Cntr=0.3,0.1

Type RM Length L Ch R = 1 ,32532   ,473,473,473
BEGIN DESCRIPTION:
PALO ALTO CREEK 47.0
END DESCRIPTION:
XS GIS Cut Line= 3
      2780407.59     10077189.88      2779872.88     10076467.67
      2779608.99      10075863.5
#Sta/Elev= 30
  4049.4 1637.95  4069.4 1637.43  4103.7 1636.78  4124.5 1634.29  4168.4 1632.16
  4203.9 1627.99    4254 1617.31  4324.9 1612.51  4395.8 1610.63  4525.3 1613.28
    4832 1614.08  4846.7 1613.38  4867.2 1609.95  4882.1 1604.64  4890.5 1599.79
  4911.4 1593.99  4975.6 1593.34    4996 1590.63  4998.7 1590.13    5002 1590.63
  5031.4 1597.91  5045.8 1599.49  5051.2 1598.67  5061.4 1600.99    5116 1601.93
  5163.6 1607.59  5220.5 1617.59  5303.6 1619.99  5424.1 1623.56  5607.3 1622.16
#Mann= 8 ,-1 , 0
  4049.4      .1       0  4069.4     .05       0  4867.2      .1       0
    4996     .07       0    5002      .1       0  5031.4     .05       0
  5163.6      .1       0  5303.6     .05       0
#XS Ineff= 2 , 0
         4835.79 1614.01
Permanent Ineff=
       F       F
Bank Sta=4882.1,5061.4
XS Rating Curve= 0 ,0
Exp/Cntr=0.3,0.1

Type RM Length L Ch R = 1 ,32059   ,452,452,452
BEGIN DESCRIPTION:
PALO ALTO CREEK 46.0
END DESCRIPTION:
XS GIS Cut Line= 3
      2780574.28     10076905.19      2780143.72     10075981.56
      2779561.94     10075572.93
#Sta/Elev= 30
    4146 1633.29  4150.5 1631.19  4167.9 1628.67  4173.4 1625.81  4190.7 1625.72
  4196.3 1623.67  4213.6 1623.02  4219.1 1620.27  4235.9 1618.58  4247.5 1615.38
  4264.9 1612.96  4316.1 1609.51  4527.4 1612.18  4738.8  1611.6    4790 1605.33
  4820.6 1603.22  4909.9 1602.04  4919.9 1600.91  4950.1 1593.88  4978.5 1591.85
  4995.6 1588.46  5018.7 1590.42  5041.3 1596.98  5052.6 1601.75  5063.4 1604.08
  5075.4 1610.01  5092.8  1612.4  5340.2 1619.65  5619.9 1621.48    5876 1620.35
#Mann= 3 , 0 , 0
    4146      .1       0  4909.9     .07       0  5052.6      .1       0
#XS Ineff= 2 , 0
         4527.84 1612.16
Permanent Ineff=
       F       F
Bank Sta=4909.9,5052.6
XS Rating Curve= 0 ,0
Exp/Cntr=0.3,0.1

Type RM Length L Ch R = 1 ,31607   ,581,581,581
BEGIN DESCRIPTION:
PALO ALTO CREEK 45.0
END DESCRIPTION:
XS GIS Cut Line= 4
      2781338.84     10076376.87      2780949.92     10076237.97
      2780338.81     10075758.81      2779742.54     10075460.67
#Sta/Elev= 30
  4173.5 1634.58  4378.5 1632.69  4521.9 1627.22    4558 1627.19  4583.5 1625.28
  4639.7 1624.93  4668.6  1621.5  4697.5 1610.27  4740.8 1607.01    4797  1600.3
  4840.3 1598.58  4910.9 1606.46  4918.7 1601.92  4925.3  1594.2  4931.7 1592.02
  4975.1 1591.58  5003.7 1587.61  5045.8 1591.25  5117.9  1592.1  5138.7 1596.36
    5174 1599.29  5274.5    1605  5316.8 1610.57  5366.1 1611.67  5405.2 1610.06
  5589.7 1612.08  5740.7 1615.17  5830.1 1619.39  5880.4 1620.27  6029.7 1620.06
#Mann= 3 , 0 , 0
  4173.5      .1       0  4918.7     .05       0    5174      .1       0
#XS Ineff= 2 , 0
         4909.92 1606.42  5367.9          1611.6
Permanent Ineff=
       F       F
Bank Sta=4918.7,5174
XS Rating Curve= 0 ,0
Exp/Cntr=0.3,0.1

Type RM Length L Ch R = 1 ,31026   ,542,542,542
BEGIN DESCRIPTION:
PALO ALTO CREEK 44.0
END DESCRIPTION:
XS GIS Cut Line= 2
       2781463.2     10075745.47      2780033.02     10075169.23
#Sta/Elev= 30
    4492 1636.43  4574.3 1633.72  4619.8 1631.34  4696.9    1626  4726.5 1625.63
  4774.8 1623.15  4833.9 1622.37  4895.9 1617.67  4911.8 1615.78  4928.3 1611.12
  4941.3 1598.65  4949.9 1591.98  4960.1 1589.93  5000.8 1585.56  5003.6 1585.06
  5006.8 1585.56  5036.2 1588.76  5048.8 1591.67  5090.1  1592.7  5126.6 1596.92
  5228.7 1593.83  5251.8 1594.23  5327.3 1598.96  5359.6 1598.49  5435.1 1607.81
    5489 1610.28  5521.3 1608.13  5843.6 1611.46  5873.2 1610.79  6033.9 1616.09
#Mann= 6 ,-1 , 0
    4492      .1       0  4574.3     .05       0  4619.8      .1       0
  4895.9     .05       0  5000.8    .035       0  5006.8     .05       0
#XS Ineff= 2 , 0
                         5489.36         1610.45
Permanent Ineff=
       F       F
Bank Sta=4941.3,5126.6
XS Rating Curve= 0 ,0
Exp/Cntr=0.3,0.1

Type RM Length L Ch R = 1 ,30484   ,559,559,559
BEGIN DESCRIPTION:
PALO ALTO CREEK 43.0
END DESCRIPTION:
XS GIS Cut Line= 3
      2781886.77     10075335.73      2781268.72     10075044.06
      2779449.26     10074974.62
#Sta/Elev= 30
  4183.2 1634.51  4409.2  1630.3  4523.1 1624.95  4678.9 1620.48  4740.8 1616.64
  4908.3 1607.37  4946.9 1604.59  4966.9 1596.77    4987 1585.78  5001.2 1583.29
  5003.9 1582.79  5007.2 1583.29    5037 1588.24    5047 1586.86    5067  1587.5
    5077  1593.5    5087 1594.63  5101.1 1594.84  5157.1 1597.63  5197.1 1595.89
  5257.2 1596.87  5357.2 1606.23  5417.3 1608.77  5457.3 1606.27  5847.6 1612.84
  6037.7 1611.56    6398  1613.4  6610.7 1618.24  6628.2 1620.17  6687.4 1621.45
#Mann= 7 ,-1 , 0
  4183.2      .1       0  4740.8     .16       0  4908.3      .1       0
  5001.2     .07       0  5007.2      .1       0  5101.1     .05       0
  6610.7      .1       0
#XS Ineff= 2 , 0
                         5418.38          1608.4
Permanent Ineff=
       F       F
Bank Sta=4966.9,5087
XS Rating Curve= 0 ,0
Exp/Cntr=0.3,0.1

Type RM Length L Ch R = 1 ,29925   ,607,607,607
BEGIN DESCRIPTION:
PALO ALTO CREEK 42.0
END DESCRIPTION:
XS GIS Cut Line= 2
      2781893.74     10074641.29      2779881.65     10074197.24
#Sta/Elev= 30
  4268.8 1630.55  4458.5 1624.79  4540.5 1621.13  4612.1 1614.94  4693.6 1611.15
  4791.2  1603.6    4840 1598.54  4868.2 1592.68  4927.4 1591.59  4932.5 1591.54
  4976.2 1584.67  5016.9 1583.92  5019.6 1583.42  5022.9 1583.92  5042.2 1587.83
    5050 1587.96  5073.8  1590.1  5083.2 1592.64  5117.5 1598.16  5134.4  1603.2
  5208.3 1605.06  5346.1 1606.25  5470.9 1610.59  5531.1 1612.96  5728.4 1613.67
  5750.5 1612.77  5949.9 1614.75  6148.2 1620.53  6301.8 1622.78  6329.3 1624.22
#Mann= 8 ,-1 , 0
  4268.8     .16       0  4927.4      .1       0  5016.9     .07       0
  5022.9      .1       0    5050     .05       0  5208.3      .1       0
  5470.9     .05       0  5750.5      .1       0
Bank Sta=4932.5,5042.2
XS Rating Curve= 0 ,0
Exp/Cntr=0.3,0.1

Type RM Length L Ch R = 1 ,29318   ,852,852,852
BEGIN DESCRIPTION:
PALO ALTO CREEK 41.0
END DESCRIPTION:
XS GIS Cut Line= 2
      2781963.18     10074057.96      2780200.32     10073648.47
#Sta/Elev= 30
  4360.9 1624.65  4444.3  1625.1  4550.5 1617.43  4591.6 1613.12  4726.5 1606.02
  4800.8 1600.99  4891.1 1592.66  4920.1 1586.32  4933.8 1585.95  4961.2 1582.44
  4999.3 1581.89    5002 1581.39  5005.3 1581.89  5021.6 1585.13  5061.7 1591.02
  5066.8 1590.76  5104.3 1597.76  5154.8 1601.93  5269.2 1603.57  5401.9 1608.64
  5577.4 1608.96  5690.6 1610.23  5767.8 1611.94  5823.5 1614.64  5844.1 1614.29
  5950.2 1617.78  5992.9 1620.62  6028.9 1620.57  6069.9 1622.31  6170.7 1621.66
#Mann= 10 ,-1 , 0
  4360.9     .16       0  4726.5      .1       0  4999.3     .07       0
  5005.3      .1       0  5021.6     .05       0  5154.8      .1       0
  5401.9     .05       0  5577.4      .1       0  5690.6     .05       0
  5767.8      .1       0
#XS Ineff= 2 , 0
                         5402.66         1608.67
Permanent Ineff=
       F       F
Bank Sta=4891.1,5061.7
XS Rating Curve= 0 ,0
Exp/Cntr=0.3,0.1

Type RM Length L Ch R = 1 ,28466   ,674,674,674
BEGIN DESCRIPTION:
PALO ALTO CREEK 40.0
END DESCRIPTION:
XS GIS Cut Line= 3
      2782115.96     10073099.62      2780997.88     10073099.62
      2780400.69     10073439.88
#Sta/Elev= 30
  4337.8 1610.44  4465.3 1611.11  4665.3  1601.3  4855.3 1600.06  4955.3 1587.81
  4975.3 1580.52  4992.3 1578.08    4995 1577.58  4998.3 1578.08  5015.3 1578.86
  5029.6 1581.98  5035.3 1583.13  5075.3 1582.81  5095.3 1588.33  5195.3 1599.73
  5224.2 1600.15  5325.3 1602.08  5708.4 1602.93  5784.7 1604.75  5817.7 1606.47
  5833.6 1604.36  5839.3 1600.65  5847.2 1600.69  5855.2 1599.72  5860.9 1604.28
  5869.5 1605.05  5882.5 1609.87  5901.2 1611.17  6013.2 1615.96  6143.2 1619.49
#Mann= 9 ,-1 , 0
  4337.8      .1       0  4992.3     .07       0  4998.3      .1       0
  5029.6     .05       0  5224.2      .1       0  5784.7     .05       0
  5847.2      .1       0  5901.2     .16       0  6013.2      .1       0
#XS Ineff= 2 , 0
                         5812.27         1606.21
Permanent Ineff=
       F       F
Bank Sta=4955.3,5095.3
XS Rating Curve= 0 ,0
Exp/Cntr=0.3,0.1

Type RM Length L Ch R = 1 ,27792   ,372,372,372
BEGIN DESCRIPTION:
PALO ALTO CREEK 38.0
END DESCRIPTION:
XS GIS Cut Line= 3
      2782240.92     10072689.89      2781213.16     10072328.79
       2780034.9      10072689.2
#Sta/Elev= 30
  4231.3 1608.73  4269.1 1608.88  4371.7 1609.38  4626.8  1599.4  4662.7 1598.77
    4797 1598.36  4897.4 1589.05  4902.7 1589.59  4959.4 1583.18  4985.1 1576.53
  5004.6 1576.17  5007.4 1575.67  5010.6 1576.17  5021.4 1576.92  5052.3 1583.18
  5060.6 1586.61  5092.4 1590.46  5114.3 1591.74    5156 1597.53  5179.5 1598.33
  5439.6 1600.99  5597.8 1600.03  5877.9 1601.44  6006.8 1602.14  6072.9 1601.85
    6227  1605.5  6312.8 1609.64  6378.4 1616.99  6436.2 1620.73  6552.8 1624.39
#Mann= 15 ,-1 , 0
  4231.3      .1       0  4269.1     .05       0  4626.8      .1       0
  4662.7     .05       0    4797      .1       0  5004.6     .07       0
  5010.6      .1       0  5021.4     .05       0  5179.5      .1       0
  5439.6     .05       0  5597.8      .1       0  5877.9     .05       0
  6006.8      .1       0    6227     .16       0  6436.2     .05       0
#XS Ineff= 2 , 0
                         5844.62         1601.85
Permanent Ineff=
       F       F
Bank Sta=4902.7,5092.4
XS Rating Curve= 0 ,0
Exp/Cntr=0.3,0.1

Type RM Length L Ch R = 1 ,27420   ,150,150,150
BEGIN DESCRIPTION:
PALO ALTO CREEK 39.0
END DESCRIPTION:
XS GIS Cut Line= 2
      2782192.31     10072405.17      2780588.16     10071578.78
#Sta/Elev= 30
  4256.9 1604.39  4385.4 1599.47  4490.6 1598.01  4623.6 1598.64  4690.1 1600.15
  4767.4 1599.41    4884 1593.89  4928.3 1590.06  4958.7 1585.47    4967 1582.47
  4972.6 1582.97  4981.2 1578.65  4989.2  1576.1  5000.7 1576.06  5003.4 1575.56
  5006.7 1576.06  5011.3 1577.01  5039.1 1577.66  5144.3 1588.84  5166.5 1589.68
  5205.2 1593.12  5255.2 1593.87  5284.9 1591.62  5307.4 1586.91  5321.7 1586.28
  5397.4 1591.47  5454.7 1598.18    5715  1612.3  5858.6 1617.67  6061.4 1621.57
#Mann= 3 ,-1 , 0
  4256.9     .05       0  5000.7     .04       0  5006.7     .05       0
#XS Ineff= 2 , 0
         4713.42 1600.29 5242.44          1593.7
Permanent Ineff=
       F       F
Bank Sta=4928.3,5144.3
XS Rating Curve= 0 ,0
Exp/Cntr=0.3,0.1

Type RM Length L Ch R = 1 ,27270   ,452,452,452
BEGIN DESCRIPTION:
Mapping XS f68fc835
END DESCRIPTION:
XS GIS Cut Line= 2
      2782220.12     10072294.07      2780595.12     10071419.07
#Sta/Elev= 30
  4202.1 1601.74  4236.8 1600.25  4295.8 1598.81  4462.3 1598.03  4588.7 1599.17
  4624.2    1601  4874.1 1597.27  4942.2 1585.42  4949.7 1582.03  4955.4 1582.54
  4971.6 1577.71  5018.7 1575.32  5021.5 1574.82  5024.7 1575.32  5062.5 1578.43
  5103.1 1580.38  5141.2    1586    5172 1586.38  5201.2 1586.97  5223.1 1579.67
  5237.5 1577.96  5260.2 1581.87  5272.6 1588.49  5282.9 1590.68  5364.4 1593.35
  5397.2 1594.65  5478.8 1598.22  5578.2 1601.62  5819.4 1616.06  6047.7 1622.19
#Mann= 11 ,-1 , 0
  4202.1     .05       0  4236.8      .1       0  4295.8     .05       0
  4462.3      .1       0  5018.7     .07       0  5024.7      .1       0
  5062.5     .05       0    5172      .1       0  5364.4     .05       0
  5397.2      .1       0  5478.8     .05       0
Bank Sta=4942.2,5141.2
XS Rating Curve= 0 ,0
Exp/Cntr=0.3,0.1

Type RM Length L Ch R = 1 ,26818   ,428,428,428
BEGIN DESCRIPTION:
Mapping XS a0b29110
END DESCRIPTION:
XS GIS Cut Line= 3
      2782338.15     10072273.22      2781511.77     10071537.12
      2780672.47     10071245.79
#Sta/Elev= 30
  3762.3  1604.4    3895 1599.19  3900.6 1599.02    3987 1597.52  4190.7 1598.25
  4310.5 1598.91  4512.1 1599.09  4664.2 1596.92    4732 1596.62  4817.3 1591.35
  4859.5 1591.15  4873.4 1589.58  4883.1 1585.52  4891.5  1583.5  4896.7 1584.24
  4922.6 1576.46  4996.5 1575.26  4999.2 1574.76  5002.5 1575.26  5041.8 1579.58
  5047.1 1578.62    5063 1584.71  5110.3 1589.57  5132.1 1593.06  5140.5 1595.75
  5166.3 1596.19  5213.2 1601.31  5290.8 1608.42  5472.3 1616.79  5757.4 1622.16
#Mann= 13 ,-1 , 0
  3762.3     .05       0    3895      .1       0  3900.6     .05       0
    3987      .1       0  4190.7     .05       0  4310.5      .1       0
  4664.2     .05       0  4859.5      .1       0  4996.5     .07       0
  5002.5      .1       0  5110.3     .05       0  5132.1      .1       0
  5213.2     .05       0
Bank Sta=4873.4,5063
XS Rating Curve= 0 ,0
Exp/Cntr=0.3,0.1

Type RM Length L Ch R = 1 ,26390   ,1148,1148,1148
BEGIN DESCRIPTION:
PALO ALTO CREEK 36.0
END DESCRIPTION:
XS GIS Cut Line= 4
      2783580.58     10072757.57      2783434.76     10072377.37
      2781252.46     10071007.58      2780163.95     10070991.96
#Sta/Elev= 30
  2170.5 1602.43  2215.2 1599.66  2491.7 1601.09  2614.2 1599.57  2962.9 1603.56
  3136.8 1594.09  3179.2 1594.14  3200.4  1598.2  3236.9 1594.76  3465.2 1595.66
  3507.9 1595.93  3621.3 1595.34  3663.9 1595.69    3743 1596.52  4346.8 1596.91
  4602.4  1592.2  4760.3 1585.97    4818 1579.88  4865.1 1579.65  4990.7 1573.95
  4993.4 1573.45  4996.7 1573.95  5021.8 1578.14  5037.1 1588.76    5042 1592.21
  5064.5 1605.94  5110.2 1610.21  5618.3 1618.78  5930.3 1619.57  6242.9 1625.31
#Mann= 13 ,-1 , 0
  2170.5      .1       0  2491.7     .16       0  2614.2      .1       0
  3465.2     .05       0  3507.9      .1       0  3621.3     .05       0
  3663.9      .1       0    3743     .05       0  4865.1      .1       0
  4990.7     .07       0  4996.7      .1       0    5042     .05       0
  5930.3      .1       0
#XS Ineff= 2 , 0
         4122.13  1597.9
Permanent Ineff=
       F       F
Bank Sta=4760.3,5037.1
XS Rating Curve= 0 ,0
Exp/Cntr=0.3,0.1

Type RM Length L Ch R = 1 ,25242   ,986,986,986
BEGIN DESCRIPTION:
PALO ALTO CREEK 34.0
END DESCRIPTION:
XS GIS Cut Line= 3
      2783708.33     10072274.89      2781859.35     10069974.52
      2780626.69      10069531.8
#Sta/Elev= 30
  2558.5 1596.31  2814.7 1599.51  3037.1 1601.79  3278.3 1591.67  3305.5  1588.6
  3497.5 1595.51  4391.8 1594.66  4820.7 1589.36  4884.7 1585.04  4920.7 1582.33
  4948.7 1575.98  5003.3 1570.85    5006 1570.35  5009.3 1570.85    5049 1571.99
  5070.3 1580.23  5113.1 1584.45  5148.7 1586.03  5155.1 1588.84  5220.5 1594.83
  5237.9 1595.62  5361.5 1606.93  5411.1 1609.04  5474.2 1608.32  5513.6 1607.51
  5652.1 1607.01  5704.1 1607.48    6064 1618.66  6416.9 1618.61  6819.6 1624.51
#Mann= 12 ,-1 , 0
  2558.5      .1       0  2814.7     .05       0  3037.1      .1       0
  4391.8     .05       0  5003.3    .035       0  5009.3     .05       0
  5220.5      .1       0  5237.9     .05       0  5474.2      .1       0
  5513.6     .05       0  5652.1      .1       0  5704.1     .05       0
#XS Ineff= 2 ,-1
  2558.5 3045.79 1601.99 3107.67 4246.29 1595.86
Permanent Ineff=
       F       F
Bank Sta=4884.7,5113.1
XS Rating Curve= 0 ,0
Exp/Cntr=0.3,0.1

Type RM Length L Ch R = 1 ,24256   ,958,958,958
BEGIN DESCRIPTION:
PALO ALTO CREEK 31.0
END DESCRIPTION:
XS GIS Cut Line= 3
      2784368.05     10072795.74      2783335.05     10070200.21
      2781920.15     10068655.11
#Sta/Elev= 30
  1476.6 1612.36  1617.9 1610.14  1754.6 1603.43  1869.6 1594.01  1899.3    1599
  1930.8 1591.22  1984.6 1589.84    2687 1592.32  3140.1 1588.33  3642.1 1592.58
  4027.6 1607.95  4166.5 1606.15    4473 1595.69  4582.8 1591.51  4717.4 1584.55
  4852.6 1583.74    4966 1568.78  5005.6  1567.8  5008.3  1567.3  5011.6  1567.8
    5037 1576.19  5093.1  1584.2  5135.6 1594.63  5183.1 1597.01  5342.5 1601.91
  5370.7 1602.48  5428.2 1603.78  5710.6 1605.95  5837.4 1604.72  6365.2 1610.86
#Mann= 16 ,-1 , 0
  1476.6      .1       0  1617.9     .16       0  1754.6     .05       0
    2687      .1       0  4166.5     .16       0    4473      .1       0
  4582.8     .05       0  4717.4      .1       0  5005.6     .07       0
  5011.6      .1       0  5183.1     .05       0  5342.5      .1       0
  5370.7     .05       0  5428.2      .1       0  5710.6     .16       0
  5837.4      .1       0
#XS Ineff= 2 , 0
         4036.28 1607.24
Permanent Ineff=
       F       F
Bank Sta=4852.6,5093.1
XS Rating Curve= 0 ,0
Exp/Cntr=0.3,0.1

Type RM Length L Ch R = 1 ,23298   ,688,688,688
BEGIN DESCRIPTION:
PALO ALTO CREEK 30.0
END DESCRIPTION:
XS GIS Cut Line= 4
      2784871.51     10072908.54      2783968.73     10069974.52
      2783361.09     10068429.38      2783144.08     10068273.13
#Sta/Elev= 30
  1088.2 1616.02  1253.5 1613.08  1396.6 1602.95  1569.5 1604.92  1616.4 1607.61
  1647.8 1600.22  1710.5 1601.84  1780.7 1593.97  1951.2 1586.51  3054.4 1589.37
  3321.2 1586.66  3792.6 1590.51    4033 1600.61  4148.3 1604.89  4293.2 1601.44
  4315.5 1600.82  4585.2 1590.83  4766.4 1579.03  4799.5 1578.59  4972.5 1565.92
  4975.2 1565.42  4978.5 1565.92    5046 1567.84  5093.7 1577.81  5145.5 1584.98
    5233 1591.11  5446.7 1596.64    5476 1597.59  5749.2 1601.34  6085.7 1604.39
#Mann= 14 ,-1 , 0
  1088.2      .1       0  1569.5     .16       0  1780.7     .05       0
    4033      .1       0  4293.2     .16       0  4315.5      .1       0
  4585.2     .16       0  4766.4      .1       0  4972.5     .07       0
  4978.5      .1       0  5145.5     .16       0  5446.7      .1       0
    5476     .16       0  5749.2      .1       0
#XS Ineff= 2 , 0
         4141.48 1604.44
Permanent Ineff=
       F       F
Bank Sta=4799.5,5093.7
XS Rating Curve= 0 ,0
Exp/Cntr=0.3,0.1

Type RM Length L Ch R = 1 ,22610   ,778,778,778
BEGIN DESCRIPTION:
PALO ALTO CREEK 29.0
END DESCRIPTION:
XS GIS Cut Line= 4
       2785861.1     10072761.02      2785748.24     10071606.46
      2783994.77     10068568.27      2783222.86       10068204.
#Sta/Elev= 30
  1000.9 1611.97  1289.8 1606.24  1400.1 1599.21  1470.4 1597.61  1510.6 1593.52
  2107.6 1585.72  2324.7  1584.2  2947.1 1582.84    3612 1590.84  3722.8 1588.39
  4237.3 1600.42  4837.5 1579.74    4893    1579  4951.9 1574.08  4981.3 1565.08
  4996.1  1564.3  5001.4 1564.13  5004.2 1563.63  5007.4 1564.13  5075.4 1567.34
  5096.9 1565.52  5128.5 1574.83  5177.6 1578.89  5295.1 1585.92  5348.2  1594.6
  5572.3 1597.51  5780.5 1597.39  5908.9 1598.63  6384.2 1601.61  6522.4 1603.38
#Mann= 12 ,-1 , 0
  1000.9     .05       0  2107.6      .1       0  2324.7     .05       0
  4237.3      .1       0  4837.5     .16       0  4996.1      .1       0
  5001.4     .07       0  5007.4      .1       0  5572.3     .05       0
  5780.5      .1       0  5908.9     .05       0  6384.2      .1       0
#XS Ineff= 2 , 0
         4253.93 1600.16
Permanent Ineff=
       F       F
Bank Sta=4893,5177.6
XS Rating Curve= 0 ,0
Exp/Cntr=0.3,0.1

Type RM Length L Ch R = 1 ,21832   ,755,755,755
BEGIN DESCRIPTION:
PALO ALTO CREEK 28.0
END DESCRIPTION:
XS GIS Cut Line= 4
      2786815.93     10072023.09      2785270.81      10069358.2
      2784767.34     10068238.41      2784255.71     10067588.03
#Sta/Elev= 30
  1339.5    1618  1519.8 1606.24  1628.5 1593.59  1789.6 1584.28  2673.5  1581.8
  2860.8 1581.44  3084.4 1578.87  3121.7 1581.56  3437.3  1579.7    3641 1583.52
    3824 1581.56  4315.1 1591.84  4676.6 1579.93  4855.2    1579  4885.9 1576.58
  4901.5 1575.96  4996.6 1561.05  4999.3 1560.55  5002.6 1561.05  5038.8 1562.56
  5060.7 1570.77  5075.4 1571.89  5126.5 1572.85    5144 1576.49  5333.5 1587.83
  5349.2 1588.19  5582.8 1594.15  5948.9 1592.17  6262.7 1597.43  6475.2 1600.89
#Mann= 11 ,-1 , 0
  1339.5     .16       0  1519.8     .05       0  2673.5      .1       0
  2860.8     .05       0  4885.9      .1       0  4996.6     .07       0
  5002.6      .1       0  5075.4     .16       0  5333.5      .1       0
  5349.2     .16       0  6262.7      .1       0
#XS Ineff= 2 , 0
         4304.72 1591.77
Permanent Ineff=
       F       F
Bank Sta=4901.5,5144
XS Rating Curve= 0 ,0
Exp/Cntr=0.3,0.1

Type RM Length L Ch R = 1 ,21077   ,802,802,802
BEGIN DESCRIPTION:
PALO ALTO CREEK 26.0
END DESCRIPTION:
XS GIS Cut Line= 3
      2787779.48     10070035.27       2786078.1     10068993.61
      2784828.76     10067457.96
#Sta/Elev= 30
  2446.9 1589.63  2695.2 1587.81  2810.5 1584.97  3052.5 1577.32  3206.2 1576.33
  3373.6 1574.28  3409.6 1570.42  3484.1 1575.21  3611.5 1576.06  3874.7 1574.58
  3990.8 1574.07  4137.7  1583.6  4385.8 1588.99  4605.2 1587.75  4939.2 1570.62
  4974.4 1562.16  5000.1 1559.74  5002.9 1559.24  5006.1 1559.74  5110.1 1569.56
  5130.7 1570.56    5241 1576.31  5348.8 1577.04  5407.2 1579.64  5480.2 1582.58
  5611.6 1587.54  5704.1 1588.66  5763.5 1589.12  5830.7 1590.22  6421.5 1601.92
#Mann= 20 ,-1 , 0
  2446.9     .05       0  2695.2     .16       0  2810.5     .05       0
  3206.2      .1       0  3484.1     .16       0  3611.5      .1       0
  3874.7     .16       0  4137.7      .1       0  4385.8     .05       0
  5000.1     .07       0  5006.1      .1       0  5130.7     .16       0
    5241      .1       0  5348.8     .16       0  5407.2      .1       0
  5480.2     .16       0  5611.6     .16       0  5704.1      .1       0
  5763.5     .16       0  5830.7      .1       0
#XS Ineff= 2 , 0
         4445.59 1589.34
Permanent Ineff=
       F       F
Bank Sta=4939.2,5110.1
XS Rating Curve= 0 ,0
Exp/Cntr=0.3,0.1

Type RM Length L Ch R = 1 ,20275   ,855,855,855
BEGIN DESCRIPTION:
Mapping XS 26b6c2d9
END DESCRIPTION:
XS GIS Cut Line= 3
      2787701.34      10068637.7      2785479.15     10067708.89
      2784602.94      10067214.4
#Sta/Elev= 30
  3479.7  1589.2  3569.5 1588.94  3708.7 1581.66  3927.2 1570.09  3943.6 1566.01
  4097.3 1571.25  4622.1 1571.47  4847.2    1575    4924 1573.13    4946 1569.44
  4967.7 1563.37  4997.2 1559.55  4999.9 1559.05  5003.2 1559.55  5043.5  1559.6
  5088.5 1561.39  5119.4 1568.88  5229.2  1573.7  5346.5 1573.25  5349.2 1573.21
  5433.7 1572.31  5559.3 1576.43  5686.3 1582.91  5752.4 1586.09  5874.4 1590.71
  6015.8 1596.82  6222.8  1601.5  6294.7 1602.04  6565.9 1602.33  6894.3 1604.66
#Mann= 15 ,-1 , 0
  3479.7     .05       0  3708.7      .1       0  4997.2     .07       0
  5003.2      .1       0  5043.5     .05       0  5229.2      .1       0
  5346.5     .05       0  5349.2      .1       0  5559.3     .05       0
  5686.3      .1       0  5752.4     .05       0  5874.4      .1       0
  6222.8     .05       0  6294.7      .1       0  6565.9     .16       0
#XS Ineff= 2 , 0
         4862.72 1575.07  5281.8         1574.44
Permanent Ineff=
       F       F
Bank Sta=4946,5119.4
XS Rating Curve= 0 ,0
Exp/Cntr=0.3,0.1

Type RM Length L Ch R = 1 ,19420   ,1253,1253,1253
BEGIN DESCRIPTION:
PALO ALTO CREEK 25.0
END DESCRIPTION:
XS GIS Cut Line= 2
      2787497.92     10067509.35      2784914.52     10066856.56
#Sta/Elev= 30
  3944.2 1586.99  4350.3 1581.56    4523 1576.49  4673.1  1570.7  4773.7 1569.29
  4877.7 1569.75  4902.9 1567.45  4922.4 1558.77  4933.8 1557.28  4992.7 1556.34
  4995.4 1555.84  4998.7 1556.34  5050.6 1560.93  5067.9 1565.38  5086.5 1567.67
  5232.9 1571.41  5325.8 1568.71  5377.8 1569.13  5478.5 1574.86  5487.6 1575.49
    5532 1578.29  5589.9  1584.6  5694.1 1592.35  5780.5 1597.16  6066.3 1598.37
  6263.7 1595.73  6399.7 1594.16  6485.2 1595.04  6585.9 1597.93  6608.8 1598.23
#Mann= 17 ,-1 , 0
  3944.2     .05       0  4350.3      .1       0    4523     .05       0
  4673.1     .16       0  4773.7      .1       0  4877.7     .05       0
  4992.7    .035       0  4998.7     .05       0  5377.8      .1       0
  5478.5     .05       0  5487.6      .1       0  5589.9     .16       0
  5694.1      .1       0  5780.5     .05       0  6263.7      .1       0
  6485.2     .05       0  6585.9     .16       0
#XS Ineff= 2 , 0
                         5238.78         1571.48
Permanent Ineff=
       F       F
Bank Sta=4902.9,5086.5
XS Rating Curve= 0 ,0
Exp/Cntr=0.3,0.1

Type RM Length L Ch R = 1 ,18167   ,636,636,636
BEGIN DESCRIPTION:
Mapping XS 14523563
END DESCRIPTION:
XS GIS Cut Line= 4
      2787154.49     10067205.42      2786824.63     10066363.41
      2786642.34     10066111.67      2785366.27     10065590.83
#Sta/Elev= 30
    3562  1576.9  3689.7 1571.52  3922.4 1566.28  4186.7 1568.73  4302.3 1565.21
  4445.2 1568.14  4449.3 1568.16  4585.4 1569.46  4763.3 1564.67  4819.8    1565
  4846.1 1563.51  4863.3 1565.25  4900.1 1562.06  4916.8 1557.11  4996.7 1554.51
  4999.4 1554.01  5002.7 1554.51  5029.7 1557.66  5062.1 1569.62  5232.2 1568.18
  5390.8 1570.08  5505.5 1575.06  5632.4 1584.43  5667.2 1586.49  5753.4 1596.24
  5819.7 1598.64  5924.4 1601.63  6057.2  1605.3  6112.8  1607.1  6155.4 1608.86
#Mann= 15 ,-1 , 0
    3562      .1       0  3689.7     .05       0  4445.2      .1       0
  4449.3     .16       0  4819.8      .1       0  4996.7     .07       0
  5002.7      .1       0  5390.8     .16       0  5505.5      .1       0
  5632.4     .05       0  5667.2      .1       0  5819.7     .05       0
  5924.4      .1       0  6057.2     .05       0  6112.8      .1       0
Bank Sta=4863.3,5062.1
XS Rating Curve= 0 ,0
Exp/Cntr=0.3,0.1

Type RM Length L Ch R = 1 ,17531   ,864,864,864
BEGIN DESCRIPTION:
Mapping XS feb1d08e
END DESCRIPTION:
XS GIS Cut Line= 3
      2787194.87     10067213.56      2786858.67       10066297.
      2786514.54     10064808.44
#Sta/Elev= 30
  3164.5 1578.35  3263.5 1574.05  3397.1 1568.47  3544.3 1566.02  3838.6 1568.32
  3941.9 1564.73  4155.2 1568.88  4277.6 1569.83  4359.2  1567.4  4441.8 1566.23
  4513.6 1559.25  4652.2 1554.88  4729.2 1557.64    4760 1562.44    4801 1557.01
  4836.6 1557.12  4893.4 1558.15  5006.4 1553.33  5009.2 1552.83  5012.4 1553.33
  5016.5 1553.77  5026.3 1555.17  5088.4 1567.44  5174.9 1567.17    5332 1568.32
  5355.3 1570.27  5386.2  1576.8  5416.8 1583.16  5457.9 1586.11  5668.6 1589.07
#Mann= 12 ,-1 , 0
  3164.5      .1       0  3263.5     .05       0  4155.2     .16       0
  4359.2     .05       0  4836.6      .1       0  5006.4     .07       0
  5012.4      .1       0  5016.5     .05       0  5026.3      .1       0
  5174.9     .05       0    5332     .16       0  5386.2      .1       0
Bank Sta=4441.8,5088.4
XS Rating Curve= 0 ,0
Exp/Cntr=0.3,0.1

Type RM Length L Ch R = 1 ,16667   ,257,257,257
BEGIN DESCRIPTION:
Mapping XS 902bc20d
END DESCRIPTION:
XS GIS Cut Line= 5
      2787254.33     10067222.81      2786967.86     10066454.55
      2787072.03     10066037.89        2787427.     10065756.69
      2787571.08     10065172.36
#Sta/Elev= 30
  3506.1 1579.57  3564.8 1577.12    3761 1568.86  3912.6 1565.94  4145.5 1568.23
  4255.1 1567.62  4323.8 1564.42    4390 1565.69  4481.5 1567.92  4596.4 1567.01
  4618.9 1567.49  4680.7 1570.47  4705.6 1569.19  4855.1 1566.46  4912.8  1557.8
  4944.6 1555.63  4973.9 1552.65  4976.7 1552.15  4979.9 1552.65  5026.6 1554.03
    5033 1555.89  5047.4 1567.15  5055.5 1576.12  5069.9  1580.6  5110.4 1579.97
  5183.7 1582.66  5248.3 1582.25  5355.6 1578.65    5659 1579.73  5810.2 1578.72
#Mann= 12 ,-1 , 0
  3506.1      .1       0  3564.8     .05       0    4390      .1       0
  4596.4     .05       0  4618.9      .1       0  4705.6     .05       0
  4944.6      .1       0  4973.9     .07       0  4979.9      .1       0
  5110.4     .16       0  5248.3      .1       0    5659     .05       0
Bank Sta=4855.1,5047.4
XS Rating Curve= 0 ,0
Exp/Cntr=0.3,0.1

Type RM Length L Ch R = 1 ,16410   ,593,593,593
BEGIN DESCRIPTION:
PALO ALTO CREEK 24.0
END DESCRIPTION:
XS GIS Cut Line= 3
      2787394.98     10067205.53      2787102.81     10066597.17
      2787611.09     10065592.62
#Sta/Elev= 30
    3801 1580.52    4197 1565.69  4287.6 1564.85  4474.3 1567.86    4701 1563.73
  4748.7 1563.72  4838.4 1566.91  4893.5 1564.51  4905.6 1562.83  4915.8 1560.89
  4921.4  1557.1    4928 1554.82  4993.4  1552.4  5001.9 1552.31  5004.6 1551.81
  5007.9 1552.31  5049.5 1554.32  5055.1 1556.19  5071.7 1557.57    5094 1562.08
  5099.6 1571.64  5107.3 1575.78  5121.9 1580.59  5183.2 1582.76  5306.5 1582.61
  5348.2 1582.11  5443.6 1580.46  5472.8 1581.47  5598.5 1580.99  5601.7 1580.99
#Mann= 8 ,-1 , 0
    3801     .05       0    4701      .1       0  4993.4     .16       0
  5001.9     .07       0  5007.9     .16       0  5306.5     .05       0
  5348.2      .1       0  5598.5     .05       0
Bank Sta=4905.6,5094
XS Rating Curve= 0 ,0
Exp/Cntr=0.3,0.1

Type RM Length L Ch R = 1 ,15817   ,608,608,608
BEGIN DESCRIPTION:
PALO ALTO CREEK 23.0
END DESCRIPTION:
XS GIS Cut Line= 2
      2787886.78       10067308.      2787740.94      10065724.6
#Sta/Elev= 30
  4073.6 1581.86  4198.4 1578.75  4248.6 1576.27  4288.8 1575.56  4325.8 1573.16
  4369.1 1573.17  4435.6 1569.84  4545.3 1566.65  4660.3 1565.24  4759.8 1562.43
  4790.9 1563.11  4881.3 1561.79  4901.4  1559.3  4931.5  1553.8  4963.1 1553.08
  4998.8 1552.54  5001.5 1552.04  5004.8 1552.54    5052 1556.07  5082.1 1557.13
  5089.1 1559.27  5094.1    1559  5102.2 1560.96  5162.5 1565.19  5232.8 1565.62
  5260.6 1566.72  5343.2 1570.86  5448.2 1572.62  5632.1    1576  5663.7 1576.94
#Mann= 7 ,-1 , 0
  4073.6     .05       0  4963.1      .1       0  4998.8     .07       0
  5004.8      .1       0  5260.6     .16       0  5448.2     .05       0
  5632.1      .1       0
Bank Sta=4881.3,5102.2
XS Rating Curve= 0 ,0
Exp/Cntr=0.3,0.1

Type RM Length L Ch R = 1 ,15209   ,537,537,537
BEGIN DESCRIPTION:
PALO ALTO CREEK 22.0
END DESCRIPTION:
XS GIS Cut Line= 3
      2788518.72     10067127.43      2788345.11     10066162.12
      2787908.44     10065607.62
#Sta/Elev= 30
  4216.5 1576.15  4321.9 1573.27  4363.4 1573.04  4555.6 1566.66  4718.1 1563.79
  4799.4 1563.54  4860.4 1561.02  4880.7  1561.4    4901 1558.54  4925.3 1557.78
    4962  1553.4  4972.1 1553.97    4984 1553.21  4992.5 1550.85  4999.6 1550.38
  5002.4 1549.88  5005.6 1550.38  5022.9 1552.88  5073.7 1552.83  5104.2  1557.5
  5144.9  1558.7  5165.2 1560.71    5236 1562.66  5279.4 1562.84  5335.4 1560.67
    5358 1560.61  5601.4 1572.05  5798.9 1578.81  5848.6 1579.69  5903.1 1579.17
#Mann= 4 ,-1 , 0
  4216.5     .05       0  4999.6     .04       0  5005.6     .05       0
  5601.4      .1       0
#XS Ineff= 2 , 0
                         5273.04         1562.72
Permanent Ineff=
       F       F
Bank Sta=4925.3,5104.2
XS Rating Curve= 0 ,0
Exp/Cntr=0.3,0.1

Type RM Length L Ch R = 1 ,14672   ,661,661,661
BEGIN DESCRIPTION:
PALO ALTO CREEK 21.0
END DESCRIPTION:
XS GIS Cut Line= 3
      2788983.13     10067024.09      2788852.92     10066107.43
      2787880.16       10065478.
#Sta/Elev= 30
  4001.2 1574.39  4144.5 1573.17  4281.3 1568.86  4486.4 1564.78  4627.8 1562.65
  4661.1 1563.08  4819.7 1559.92  4880.3 1555.65  4900.5 1555.18  4928.5 1552.48
  4968.1  1548.9  5010.2 1548.38    5013 1547.88  5016.2 1548.38  5049.5 1552.29
  5063.4 1551.92  5085.8 1555.64  5122.1 1556.37  5157.4 1559.53  5230.1 1560.69
  5301.6 1559.59  5330.5    1558  5387.9 1558.75  5504.1 1563.66    5533 1563.93
  5626.7 1569.78  5748.6  1573.6  5844.3 1576.63  6005.9 1578.55  6085.7 1578.31
#Mann= 8 ,-1 , 0
  4001.2     .05       0  4661.1     .16       0  4928.5      .1       0
  5010.2     .07       0  5016.2      .1       0  5157.4     .05       0
  5748.6      .1       0  6005.9     .05       0
#XS Ineff= 2 , 0
                         5221.28         1560.56
Permanent Ineff=
       F       F
Bank Sta=4900.5,5085.8
XS Rating Curve= 0 ,0
Exp/Cntr=0.3,0.1

Type RM Length L Ch R = 1 ,14011   ,287,287,287
BEGIN DESCRIPTION:
PALO ALTO CREEK 16.0
END DESCRIPTION:
XS GIS Cut Line= 3
      2790498.13     10065509.36      2789732.89      10065456.9
      2787932.15     10065447.65
#Sta/Elev= 30
  3448.8 1590.42  3545.8 1587.75  3623.9 1585.78  3729.1 1584.69  3869.4 1581.24
  4059.6 1581.01  4192.1 1579.92  4318.1  1577.1  4511.1 1569.96  4600.3 1566.84
  4727.1 1555.79  4730.3 1555.31  4770.3 1550.48  4830.3  1550.5  4840.3  1547.6
  4860.3 1549.87  4900.3 1550.19  4987.3 1546.39    4990 1545.89  4993.3 1546.39
  5003.9 1546.76  5030.3 1548.01  5070.3 1556.23  5100.3 1556.74  5170.3 1553.94
  5299.9 1559.02  5375.3 1561.67  5670.3 1571.21  5690.3 1572.88  6016.6 1578.11
#Mann= 12 ,-1 , 0
  3448.8      .1       0  3545.8     .05       0  3623.9      .1       0
  4059.6     .05       0  4318.1      .1       0  4511.1     .16       0
  4727.1      .1       0  4987.3     .07       0  4993.3      .1       0
  5003.9     .05       0  5299.9      .1       0  5375.3     .05       0
Bank Sta=4730.3,5070.3
XS Rating Curve= 0 ,0
Exp/Cntr=0.3,0.1

Type RM Length L Ch R = 1 ,13724   ,1138,1138,1138
BEGIN DESCRIPTION:
PALO ALTO CREEK 19.0
END DESCRIPTION:
XS GIS Cut Line= 2
      2789681.05     10065341.81      2787623.74      10064899.1
#Sta/Elev= 30
  4209.5 1578.27  4272.4 1576.49  4469.4 1567.94  4549.7 1563.28  4644.1 1553.98
  4662.2 1551.55  4703.9 1549.73  4754.3 1550.98    4785  1548.3  4792.3 1545.42
  4815.6  1549.1  4856.6 1550.17  4928.2 1545.33  4996.8 1544.92  4999.5 1544.42
  5002.8 1544.92  5009.8 1545.69  5028.8 1550.65  5033.9 1550.37  5050.9 1553.71
  5102.1 1552.74  5250.8 1556.26  5413.6 1560.02    5551 1564.02  5605.5 1563.74
    5634 1564.99  5649.7 1568.13    5694 1569.36  6043.1  1572.4  6313.9 1578.35
#Mann= 9 ,-1 , 0
  4209.5     .05       0  4272.4      .1       0  4469.4     .16       0
  4644.1      .1       0  4996.8     .07       0  5002.8      .1       0
  5009.8     .05       0  5250.8      .1       0  5413.6     .05       0
Bank Sta=4856.6,5028.8
XS Rating Curve= 0 ,0
Exp/Cntr=0.3,0.1

Type RM Length L Ch R = 1 ,12586   ,662,662,662
BEGIN DESCRIPTION:
PALO ALTO CREEK 18.0
END DESCRIPTION:
XS GIS Cut Line= 3
      2790309.92     10064367.67      2789060.22     10064049.84
      2787659.37     10064302.86
#Sta/Elev= 30
  3142.4 1568.65  3474.1 1560.64  3659.8 1558.87  3800.7 1554.05  3864.7 1550.56
  4000.3 1548.43  4028.4 1544.21  4069.3 1542.34  4186.1 1540.02  4206.7 1542.68
  4268.6 1542.75  4386.9 1547.79  4487.8 1549.35  4697.9  1552.1  4803.4 1546.86
    4830 1545.98  4870.6 1543.15  4901.1 1544.18  4921.4  1541.7  4951.9 1543.54
  4999.7 1537.42  5002.5 1536.92  5005.7 1537.42  5046.5 1541.91  5063.7 1548.25
  5185.6 1560.15  5297.4 1564.46  5382.9 1566.57  5553.7 1565.36  5855.4 1573.75
#Mann= 7 ,-1 , 0
  3142.4     .05       0  3800.7      .1       0  4386.9     .05       0
  4487.8     .16       0  4803.4      .1       0  4999.7     .07       0
  5005.7     .05       0
Bank Sta=4830,5063.7
XS Rating Curve= 0 ,0
Exp/Cntr=0.3,0.1

Type RM Length L Ch R = 1 ,11924   ,1106,1106,1106
XS GIS Cut Line= 2
     2790332.401    10063706.119      2787684.79    10063454.859
#Sta/Elev= 30
       0 1568.81  279.99 1559.19  339.98 1556.11  399.98 1556.28  459.98 1553.68
  509.97 1554.32  559.97 1551.68  629.97 1551.27  779.96 1546.76  909.95  1547.6
  949.95 1544.57  989.95 1539.77 1059.95 1537.61 1159.94 1538.32 1239.94 1545.12
 1289.93 1546.27 1469.92 1545.31  1869.9 1549.51  1889.9 1547.64  1949.9 1535.52
  1999.9 1534.64  2029.9  1536.6  2039.9 1538.17 2059.89 1544.15 2069.89 1545.44
 2199.89 1546.74 2279.88 1549.21 2399.88 1553.92 2569.87 1564.05 2659.86 1565.69
#Mann= 3 , 0 , 0
       0      .1       0  1889.9     .07       0 2069.89      .1       0
Bank Sta=1889.9,2069.89
XS Rating Curve= 0 ,0
Exp/Cntr=0.3,0.1

Type RM Length L Ch R = 1 ,10818   ,706,706,706
XS GIS Cut Line= 3
     2790403.654    10063124.845     2789938.635    10063192.348
     2788209.812    10062652.325
#Sta/Elev= 30
       0 1570.92  119.33 1568.52  149.16 1568.87   248.6 1565.25   338.1 1563.47
  377.88 1560.96  457.43 1558.28  547.13 1551.33  567.08 1551.12     597 1548.51
   746.6 1546.76   856.3 1547.95  946.06 1546.64  985.96 1544.04 1015.88 1543.27
  1155.5 1543.69 1225.32 1542.13 1275.18 1539.59 1374.92 1531.62 1404.84 1527.99
 1464.68 1531.08 1474.65 1532.56 1504.57 1540.49 1514.54 1541.46 1574.38 1542.06
 1634.22  1545.4 1694.06  1546.8 1953.37 1557.68 2073.05 1560.99 2282.49 1563.39
#Mann= 3 , 0 , 0
       0      .1       0 1275.18     .07       0 1504.57      .1       0
Bank Sta=1275.18,1504.57
XS Rating Curve= 0 ,0
Exp/Cntr=0.3,0.1

Type RM Length L Ch R = 1 ,10112   ,713,713,713
BEGIN DESCRIPTION:
PALO ALTO CREEK 15.0
END DESCRIPTION:
XS GIS Cut Line= 4
       2790361.3     10062478.29       2789840.5     10062326.39
      2788505.87     10062152.78      2787909.07     10062380.65
#Sta/Elev= 30
  3899.3 1569.79  3903.2 1569.79  3969.6 1566.93  4036.5 1560.71  4131.4 1556.18
  4173.1 1555.83  4233.2 1552.12  4266.8 1552.46  4397.4 1547.84  4511.5 1546.71
  4645.5 1545.23  4786.7  1540.8  4808.4 1538.76  4890.7  1536.2  4909.9 1533.58
    4938 1527.99  4966.8 1525.58  4969.6 1525.08  4972.8 1525.58  5018.7 1526.61
    5059 1535.66  5089.2 1539.88  5137.3 1542.77  5164.6 1543.21  5391.8 1545.63
    5543 1552.89  5610.6 1554.28  5802.7 1554.42  5862.8 1556.57  6426.5    1560
#Mann= 11 ,-1 , 0
  3899.3      .1       0  3903.2     .05       0  4233.2      .1       0
  4511.5     .05       0  4808.4     .16       0  4909.9      .1       0
  4966.8     .07       0  4972.8      .1       0  5137.3     .16       0
  5164.6      .1       0  5610.6     .05       0
Bank Sta=4890.7,5059
XS Rating Curve= 0 ,0
Exp/Cntr=0.3,0.1

Type RM Length L Ch R = 1 ,9399    ,614,614,614
BEGIN DESCRIPTION:
PALO ALTO CREEK 13.0
END DESCRIPTION:
XS GIS Cut Line= 2
      2790014.33     10061591.81      2787753.93     10061643.89
#Sta/Elev= 30
  4461.6 1560.55  4497.5 1560.03  4547.5 1556.79  4587.5 1556.84    4620 1554.44
  4745.3 1549.35  4787.6  1548.6  4857.6 1541.27    4871 1538.64  4917.6 1534.94
  4927.6 1533.66  4947.6 1525.54  4957.6 1523.79  4977.6  1524.9  5004.6 1523.47
  5007.4 1522.97  5010.6 1523.47  5011.3 1523.52  5107.6  1532.5  5167.7 1533.73
  5237.7 1540.53    5496  1541.7  5576.6 1544.56  5701.5 1547.93  5867.8  1546.5
  6063.7  1542.1    6308  1541.4    6458 1545.03    6528 1548.54  6722.6 1551.88
#Mann= 11 ,-1 , 0
  4461.6     .05       0    4620      .1       0  4745.3     .16       0
    4871      .1       0  5004.6     .07       0  5010.6      .1       0
  5011.3     .05       0    5496      .1       0  5576.6     .05       0
  5701.5      .1       0  5867.8     .05       0
Bank Sta=4917.6,5107.6
XS Rating Curve= 0 ,0
Exp/Cntr=0.3,0.1

Type RM Length L Ch R = 1 ,8785    ,931,931,931
BEGIN DESCRIPTION:
PALO ALTO CREEK 12.0
END DESCRIPTION:
XS GIS Cut Line= 3
      2790087.31     10061320.98      2789399.79     10061008.47
      2787738.37     10061190.76
#Sta/Elev= 30
    4140 1557.14  4317.2 1551.54  4357.9 1549.12  4415.1 1549.33  4628.2 1543.28
  4731.9 1543.13  4760.5 1541.34  4800.6 1539.59  4841.3 1534.69  4846.7 1535.77
  4863.7 1533.58  4916.7    1533  4926.5 1532.48  4982.7 1522.75  4985.4 1522.25
  4988.7 1522.75  5037.4  1523.9  5076.8 1533.53  5117.9 1539.24    5148  1540.6
  5379.4 1538.68  5731.5  1543.6  5772.7    1543  5822.1 1543.04  5842.2 1544.56
  5901.8 1541.24  6043.4 1540.92  6276.4 1545.83  6516.2 1553.94  6566.6 1554.15
#Mann= 7 ,-1 , 0
    4140     .05       0  4317.2      .1       0  4760.5     .16       0
  4926.5      .1       0  4982.7     .07       0  4988.7      .1       0
  5772.7     .05       0
#XS Ineff= 1 ,-1
 5844.62  6236.4 1544.53
Permanent Ineff=
       F
Bank Sta=4916.7,5076.8
XS Rating Curve= 0 ,0
Exp/Cntr=0.3,0.1
