--- SOUTH GRAPE CREEK.prj (project) ---

Proj Title=SOUTH GRAPE CREEK Base Level Engineering
Current Plan=p01
Default Exp/Contr=0.3,0.1
English Units
Geom File=g01
Flow File=f01
Plan File=p01
Y Axis Title=Elevation
X Axis Title(PF)=Main Channel Distance
X Axis Title(XS)=Station
BEGIN DESCRIPTION:
SOUTH GRAPE CREEK
END DESCRIPTION:
DSS File=dss
DSS Export Rating Curves= 0
DSS Export Rating Curve Sorted= 0
DSS Export Volume Flow Curves= 0
DXF OffsetX= 0
DXF OffsetY= 0
DXF ScaleX= 1
DXF ScaleY= 10

--- SOUTH GRAPE CREEK.p01 (plan) ---

Plan Title=Multiple Run
Program Version=4.10
Short Identifier=Multiple Run
Geom File=g01
Flow File=f01
Subcritical Flow
K Sum by GR= 0
Std Step Tol= 0.01
Critical Tol= 0.01
Num of Std Step Trials= 20
Max Error Tol= 0.3
Flow Tol Ratio= 0.001
Split Flow NTrial= 30
Split Flow Tol= 0.02
Split Flow Ratio= 0.02
Log Output Level= 0
Friction Slope Method= 1
Unsteady Friction Slope Method= 2
Unsteady Bridges Friction Slope Method= 1
Parabolic Critical Depth
Global Vel Dist= 1 , 1 , 1
Global Log Level= 0
CheckData=True
Encroach Param=-1 ,0,0, 0
BEGIN DESCRIPTION:
Multiple Run
END DESCRIPTION:
Computation Interval=1HOUR
Output Interval=1HOUR
Run HTab= 0
Run UNet= 0
Run PostProcess= 0
Run WQNet= 0
UNET Theta= 1
UNET Theta Warmup= 1
UNET ZTol= 0.02
UNET ZSATol= 0.05
UNET MxIter= 20
UNET MaxInSteps= 0
UNET DtIC= 0
UNET DtMin= 0
UNET MaxCRTS= 20
UNET WFStab= 2
UNET SFStab= 1
UNET WFX= 1
UNET SFX= 1
UNET DSS MLevel= 4
UNET DZMax Abort= 100
UNET Convert EG Bridges= 0
UNET Use Existing IB Tables=-1
UNET Froude Reduction=False
UNET Froude Limit= 1
UNET Froude Power= 10
UNET Time Slicing=0,0, 5
UNET Junction Losses=0
Instantaneous Interval=1HOUR
DSS File=dss
Write IC File= 0
Write IC File at Sim End=0
Echo Input=False
Echo Parameters=False
Echo Output=False
Write Detailed= 0
WQ AD Non Conservative
WQ ULTIMATE=-1
WQ Max Comp Step=1HOUR
WQ Output Interval=15MIN
WQ Output Selected Increments= 0
WQ Output face flow=0
WQ Output face velocity=0
WQ Output face area=0
WQ Output face dispersion=0
WQ Output cell volume=0
WQ Output cell surface area=0
WQ Output cell continuity=0
WQ Output cumulative cell continuity=0
WQ Output face conc=0
WQ Output face dconc_dx=0
WQ Output face courant=0
WQ Output face peclet=0
WQ Output face adv mass=0
WQ Output face disp mass=0
WQ Output cell mass=0
WQ Output cell source sink temp=0
WQ Output cell source sink nsm=0
WQ Output MaxMinRange=-1
WQ Daily Max Min Mean=-1
WQ Daily Range=0
WQ Daily Time=0
WQ Create Restart=0
WQ Fixed Restart=0
WQ System Summary=0
WQ Use Fixed Temperature=0
Sorting and Armoring Iterations= 10
XS Update Threshold= 0.02
Hydraulics Update Threshold= 0.02
Energy Slope Method= 1
Volume Change Method= 0
XS Weighting Method= 0
Number of US Weighted Cross Sections= 1
Number of DS Weighted Cross Sections= 1
Upstream XS Weight=0.25
Main XS Weight=0.5
Downstream XS Weight=0.25
Number of DS XS's Weighted with US Boundary= 1
Upstream Boundary Weight= 1
Weight of XSs Associated with US Boundary= 0
Number of US XS's Weighted with DS Boundary= 1
Downstream Boundary Weight= 0.5
Weight of XSs Associated with DS Boundary= 0.5
Sediment Output Level= 4
Mass or Volume Output= 0
Output Increment Type= 1
Profile and TS Output Increment= 10
XS Output Flag= 0
XS Output Increment= 10
Disregard all LS=0
Disregard all Conn=0
Disregard all Breaches=0
Disregard all Pumps=0

--- SOUTH GRAPE CREEK.f01 (steady flow) ---

Flow Title=Multiple
Program Version=4.10
Number of Profiles= 7
Profile Names=10-year,25-year,50-year,1pct_min,100-year,1pct_plu,500-year
River Rch & RM=SOUTH GRAPE CREE,Reach-1         ,87875
     352     484     592     533     720     974    1068
River Rch & RM=SOUTH GRAPE CREE,Reach-1         ,85742
     912    1321    1676    1555    2103    2844    3326
River Rch & RM=SOUTH GRAPE CREE,Reach-1         ,83979
    1160    1701    2174    2031    2747    3714    4404
River Rch & RM=SOUTH GRAPE CREE,Reach-1         ,79318
    1837    2754    3573    3382    4574    6186    7536
River Rch & RM=SOUTH GRAPE CREE,Reach-1         ,77274
    1984    2975    3859    3652    4938    6679    8128
River Rch & RM=SOUTH GRAPE CREE,Reach-1         ,72145
    2621    3972    5189    4941    6682    9037   11137
River Rch & RM=SOUTH GRAPE CREE,Reach-1         ,71863
    2621    3972    5189    4941    6682    9037   11137
River Rch & RM=SOUTH GRAPE CREE,Reach-1         ,66714
    2831    4301    5629    5368    7259    9817   12136
River Rch & RM=SOUTH GRAPE CREE,Reach-1         ,65943
    3200    4879    6403    6118    8274   11190   13890
River Rch & RM=SOUTH GRAPE CREE,Reach-1         ,65798
    3200    4879    6403    6118    8274   11190   13890
River Rch & RM=SOUTH GRAPE CREE,Reach-1         ,65296
    3200    4879    6403    6118    8274   11190   13890
River Rch & RM=SOUTH GRAPE CREE,Reach-1         ,60703
    4190    6450    8519    8187   11072   14974   18802
River Rch & RM=SOUTH GRAPE CREE,Reach-1         ,59971
    4190    6450    8519    8187   11072   14974   18802
River Rch & RM=SOUTH GRAPE CREE,Reach-1         ,57095
    4290    6594    8699    8350   11293   15272   19128
River Rch & RM=SOUTH GRAPE CREE,Reach-1         ,49571
    5585    8654   11481   11075   14978   20256   25618
River Rch & RM=SOUTH GRAPE CREE,Reach-1         ,48336
    5585    8654   11481   11075   14978   20256   25618
River Rch & RM=SOUTH GRAPE CREE,Reach-1         ,45307
    5793    8977   11910   11488   15537   21012   26568
River Rch & RM=SOUTH GRAPE CREE,Reach-1         ,44278
    5793    8977   11910   11488   15537   21012   26568
River Rch & RM=SOUTH GRAPE CREE,Reach-1         ,40482
    6038    9361   12422   11983   16206   21917   27718
River Rch & RM=SOUTH GRAPE CREE,Reach-1         ,35606
    6000    9283   12301   11849   16025   21672   27325
River Rch & RM=SOUTH GRAPE CREE,Reach-1         ,30112
    6853   10638   14131   13640   18447   24947   31583
River Rch & RM=SOUTH GRAPE CREE,Reach-1         ,29076
    6853   10638   14131   13640   18447   24947   31583
River Rch & RM=SOUTH GRAPE CREE,Reach-1         ,23235
    7234   11242   14945   14436   19524   26403   33472
River Rch & RM=SOUTH GRAPE CREE,Reach-1         ,21772
    9890   15457   20634   20003   27052   36585   46690
River Rch & RM=SOUTH GRAPE CREE,Reach-1         ,20918
    9890   15457   20634   20003   27052   36585   46690
River Rch & RM=SOUTH GRAPE CREE,Reach-1         ,16985
   10154   15878   21204   20563   27809   37608   48026
River Rch & RM=SOUTH GRAPE CREE,Reach-1         ,13255
   10154   15878   21204   20563   27809   37608   48026
River Rch & RM=SOUTH GRAPE CREE,Reach-1         ,12062
   10286   16059   21423   20751   28064   37953   48351
River Rch & RM=SOUTH GRAPE CREE,Reach-1         ,4112
   10258   15994   21317   20629   27898   37728   47970
Boundary for River Rch & Prof#=SOUTH GRAPE CREE,Reach-1         , 1
Up Type= 0
Dn Type= 3
Dn Slope=0.00013
Boundary for River Rch & Prof#=SOUTH GRAPE CREE,Reach-1         , 2
Up Type= 0
Dn Type= 3
Dn Slope=0.00013
Boundary for River Rch & Prof#=SOUTH GRAPE CREE,Reach-1         , 3
Up Type= 0
Dn Type= 3
Dn Slope=0.00013
Boundary for River Rch & Prof#=SOUTH GRAPE CREE,Reach-1         , 4
Up Type= 0
Dn Type= 3
Dn Slope=0.00013
Boundary for River Rch & Prof#=SOUTH GRAPE CREE,Reach-1         , 5
Up Type= 0
Dn Type= 3
Dn Slope=0.00013
Boundary for River Rch & Prof#=SOUTH GRAPE CREE,Reach-1         , 6
Up Type= 0
Dn Type= 3
Dn Slope=0.00013
Boundary for River Rch & Prof#=SOUTH GRAPE CREE,Reach-1         , 7
Up Type= 0
Dn Type= 3
Dn Slope=0.00013
DSS Import GetInterval= 0
DSS Import GetPeak= 0
DSS Import FillOption= 0

--- SOUTH GRAPE CREEK.g01 (geometry) ---

Geom Title=Existing Conditions
Program Version=4.10

River Reach=SOUTH GRAPE CREE,Reach-1
Reach XY= 30
      2763613.76     10014218.95      2764435.13     10012524.42
      2765911.15     10013287.39      2769374.25     10010265.24
      2772893.66     10011273.09      2774032.56     10010555.79
      2775812.18     10011738.19      2774728.92     10012988.35
      2776324.36     10013562.59      2776816.89     10020692.89
      2780040.04     10022779.94      2781635.42     10022518.65
      2784908.08     10025835.88      2785419.17     10027381.93
      2787373.21     10026374.44      2790314.87     10027325.91
      2790864.04      10028322.6      2791368.47     10027613.73
      2792317.73     10028206.14      2793845.28     10030315.26
      2795416.83     10030238.51      2795459.48     10034176.34
      2799562.98     10034145.12      2802443.48     10036730.81
      2803602.29     10041582.15      2804840.49     10042698.08
      2803271.08     10046302.49      2804215.79     10048472.49
      2807035.34     10050044.96      2806386.73      10052073.2

Type RM Length L Ch R = 1 ,87875   ,545,545,545
BEGIN DESCRIPTION:
SOUTH GRAPE CREEK 151.0
END DESCRIPTION:
XS GIS Cut Line= 2
       2763973.1     10014198.94      2763454.42     10013998.39
#Sta/Elev= 30
  4785.1 1923.42  4822.4 1920.35  4894.3 1916.57  4918.7 1914.48  4948.8 1903.85
  4954.2 1903.44  4961.2 1904.15  4972.3  1904.9  4978.7 1904.64  4984.1 1903.83
  5005.7 1903.25  5008.4 1902.75  5011.7 1903.25  5025.9 1904.73  5028.6 1905.42
  5033.3 1906.63  5047.4 1908.29  5093.2 1908.25  5117.7 1909.04  5123.1 1908.69
  5142.3 1909.61  5147.7 1909.17  5165.3 1910.22  5196.9  1910.6  5206.4 1911.36
  5226.8 1912.19  5232.2 1910.91  5251.1  1911.8    5294 1916.69  5341.2 1919.95
#Mann= 7 ,-1 , 0
  4785.1      .1       0  4822.4     .16       0  4961.2     .05       0
  5005.7    .035       0  5011.7     .05       0  5028.6      .1       0
  5206.4     .05       0
Bank Sta=4978.7,5025.9
XS Rating Curve= 0 ,0
Exp/Cntr=0.3,0.1

Type RM Length L Ch R = 1 ,87330   ,450,450,450
BEGIN DESCRIPTION:
SOUTH GRAPE CREEK 150.0
END DESCRIPTION:
XS GIS Cut Line= 2
      2764202.22     10013789.21      2763502.12     10013435.69
#Sta/Elev= 30
  4673.1 1926.92  4695.2 1923.46  4700.8 1923.38  4721.6 1920.34  4746.6 1918.96
  4762.1 1916.52  4778.1 1914.99  4806.7 1909.17  4845.3 1903.18  4867.8 1896.84
  4879.2 1894.36  4901.5 1893.67  4918.2 1894.47  4923.8 1894.06  4934.9 1895.24
  4957.2 1894.41  4968.6 1892.57  4979.5  1892.2  5001.5  1888.7  5004.8  1889.2
  5013.4 1892.75  5029.7 1896.32  5068.6 1898.65    5103 1902.59    5247 1909.94
  5274.9 1910.58  5349.5 1916.68  5403.1 1919.77  5420.6 1921.73  5457.4 1926.79
#Mann= 6 ,-1 , 0
  4673.1      .1       0  4721.6     .16       0  4746.6      .1       0
  4979.5     .07       0  5013.4      .1       0  5420.6     .05       0
#XS Ineff= 2 , 0
         4935.03 1895.18
Permanent Ineff=
       T       T
Bank Sta=4979.5,5013.4
XS Rating Curve= 0 ,0
Exp/Cntr=0.3,0.1

Type RM Length L Ch R = 1 ,86880   ,337,337,337
BEGIN DESCRIPTION:
SOUTH GRAPE CREEK 149.0
END DESCRIPTION:
XS GIS Cut Line= 3
       2764493.9     10013532.27      2764271.68     10013344.77
      2763598.06     10013254.49
#Sta/Elev= 30
  4595.4 1920.98    4627 1922.11  4686.8 1920.09  4797.4 1915.44  4847.6 1911.07
    4887 1908.54  4933.2  1906.4    4960 1903.83  4970.1 1902.06  4980.2    1897
  4993.6 1884.82  4997.4 1881.66  5000.1 1881.16  5003.4 1881.66  5006.2  1883.5
  5011.2 1883.35 5017.67 1884.82  5020.6  1885.5  5050.8 1886.67  5079.1 1890.53
  5111.4 1890.19  5252.6 1894.99    5303 1898.57  5308.1 1898.27  5343.4 1902.06
  5393.9 1904.17  5407.5 1905.55  5455.6 1909.91  5494.8 1915.58  5565.8  1920.1
#Mann= 9 ,-1 , 0
  4595.4      .1       0  4686.8     .16       0  4847.6      .1       0
    4887     .16       0  4993.6     .07       0  5020.6      .1       0
  5252.6      .1       0  5407.5     .16       0  5455.6      .1       0
Bank Sta=4993.6,5017.67
XS Rating Curve= 0 ,0
Exp/Cntr=0.3,0.1

Type RM Length L Ch R = 1 ,86543   ,397,397,397
BEGIN DESCRIPTION:
SOUTH GRAPE CREEK 147.0
END DESCRIPTION:
XS GIS Cut Line= 4
      2764528.62     10013358.66      2764278.62     10013087.82
      2764021.68     10012948.93      2763452.88     10013073.79
#Sta/Elev= 30
  4473.8    1913  4559.9 1910.34  4698.8 1906.07  4732.2 1903.69  4841.8 1890.18
  4876.7 1888.16  4898.6 1883.23  4904.3 1883.67  4920.5 1880.94  4933.5 1881.22
  4942.4 1878.39  4964.3 1877.09    4970 1879.39    4979 1877.22  4998.7  1874.5
  5001.5    1874  5004.7  1874.5  5013.7 1877.76  5024.2 1883.68  5028.7 1884.22
  5046.1 1885.63  5138.7 1885.67    5267 1891.57    5369 1900.22    5471 1909.06
  5516.6 1914.77    5573 1917.56  5576.5 1917.72  5665.7 1927.67  5716.8 1930.02
#Mann= 12 ,-1 , 0
  4473.8      .1       0  4559.9     .16       0  4698.8      .1       0
  4998.7     .07       0  5004.7      .1       0  5028.7     .05       0
    5267     .16       0    5369      .1       0    5471     .05       0
    5573      .1       0  5576.5     .05       0  5665.7      .1       0
Bank Sta=4979,5013.7
XS Rating Curve= 0 ,0
Exp/Cntr=0.3,0.1

Type RM Length L Ch R = 1 ,86146   ,404,404,404
BEGIN DESCRIPTION:
SOUTH GRAPE CREEK 148.0
END DESCRIPTION:
XS GIS Cut Line= 4
      2764459.18     10013233.65      2764452.23     10012733.66
      2764174.46      10012678.1      2763473.23     10013011.35
#Sta/Elev= 30
  4388.1 1908.53    4438 1906.53    4508 1896.69    4698 1878.66  4801.2 1876.99
  4885.6 1873.94  4973.6 1875.31 4985.86 1872.99    4994 1869.11  5001.2 1868.56
  5003.9 1868.06  5007.2 1868.56  5011.8 1873.03  5034.8 1875.74  5063.2 1876.25
  5095.9 1874.71  5119.3 1875.77  5146.9    1879  5190.9 1878.55  5385.8 1880.62
  5428.2 1882.33  5475.8 1886.84    5519 1889.02  5585.9 1894.84  5720.6 1906.41
    5796 1915.05  5810.4 1915.73  5870.9 1918.59  5921.9  1925.5  5947.8 1928.16
#Mann= 11 ,-1 , 0
  4388.1     .16       0    4438      .1       0  5001.2     .07       0
  5007.2      .1       0  5190.9     .16       0  5385.8      .1       0
  5475.8     .05       0  5585.9      .1       0    5796     .05       0
  5810.4      .1       0  5921.9     .05       0
#XS Ineff= 2 , 0
         4962.65 1875.61 5063.37         1876.21
Permanent Ineff=
       T       T
Bank Sta=4985.86,5011.8
XS Rating Curve= 0 ,0
Exp/Cntr=0.3,0.1

Type RM Length L Ch R = 1 ,85742   ,507,507,507
BEGIN DESCRIPTION:
SOUTH GRAPE CREEK 146.0
END DESCRIPTION:
XS GIS Cut Line= 3
      2764577.23     10013282.25      2764639.73     10012080.88
      2764459.19     10011719.79
#Sta/Elev= 30
  4255.6 1910.36  4309.4 1904.69  4368.2 1897.94  4404.3 1892.61  4464.4 1887.49
  4524.5 1878.63  4549.5 1876.94  4604.6 1874.34  4760.2 1874.26  4913.8 1868.95
    4935 1869.83  4975.1 1865.78  4992.1 1860.44  4994.9 1859.94  4998.1 1860.44
  5015.1 1862.36  5025.2 1866.29    5041 1869.08  5115.3 1879.19  5142.9 1887.89
  5147.9 1888.04  5195.4 1907.51  5237.6 1917.01  5345.6 1941.18  5415.7 1949.28
    5478 1961.89  5534.6 1966.31  5552.2 1968.13  5679.2 1971.34  5862.3 1971.11
#Mann= 11 ,-1 , 0
  4255.6      .1       0  4309.4     .16       0  4368.2      .1       0
  4549.5     .05       0  4913.8      .1       0  4992.1     .07       0
  4998.1      .1       0    5041     .16       0  5237.6      .1       0
  5534.6     .05       0  5552.2      .1       0
Bank Sta=4975.1,5025.2
XS Rating Curve= 0 ,0
Exp/Cntr=0.3,0.1

Type RM Length L Ch R = 1 ,85235   ,397,397,397
BEGIN DESCRIPTION:
SOUTH GRAPE CREEK 145.0
END DESCRIPTION:
XS GIS Cut Line= 2
      2764674.47     10013185.03       2765326.6     10012408.02
#Sta/Elev= 30
  4374.4 1892.63  4399.8 1889.14  4406.3 1889.74    4435 1884.18  4455.8 1882.62
  4493.3 1877.09  4532.7  1871.7  4562.4  1869.1  4593.6 1868.31  4761.5 1867.11
  4860.4 1863.01  4924.4 1863.48    4952 1861.47  4974.8 1861.09  4981.3 1855.78
  4992.6 1853.61  4995.4 1853.11  4998.6 1853.61  5009.9 1855.65  5016.5 1860.48
  5024.2 1864.83  5030.8 1866.56  5067.2 1872.51  5130.9 1877.84  5172.6 1878.36
  5215.5 1880.99  5250.8 1887.15  5336.5 1906.61  5385.9 1915.38  5388.8  1917.4
#Mann= 7 ,-1 , 0
  4374.4      .1       0  4493.3     .16       0  4532.7      .1       0
  4593.6     .05       0    4952      .1       0  4992.6     .07       0
  4998.6      .1       0
Bank Sta=4974.8,5016.5
XS Rating Curve= 0 ,0
Exp/Cntr=0.3,0.1

Type RM Length L Ch R = 1 ,84838   ,402,402,402
BEGIN DESCRIPTION:
SOUTH GRAPE CREEK 144.0
END DESCRIPTION:
XS GIS Cut Line= 3
      2764959.15     10013351.74      2765535.57     10012816.99
      2765625.83     10012539.25
#Sta/Elev= 30
  4460.3 1889.69  4479.6 1885.71  4493.8 1886.23  4500.6 1884.16    4508 1884.19
  4571.5 1873.15  4628.2 1867.71  4684.9 1867.42  4840.7 1859.11  4911.1 1858.43
  4932.6 1855.57  4967.8 1857.46  4975.1 1856.78  4995.9 1852.04  5010.3 1853.32
  5024.5 1857.55  5038.6 1859.93  5095.3 1859.19  5208.7 1861.37  5274.2    1864
  5323.6 1869.22    5370 1870.71    5402 1875.13  5418.2 1880.22  5433.9 1881.31
  5439.3 1884.45  5465.9 1892.12  5523.4 1903.29  5529.8 1905.64  5538.6 1905.95
#Mann= 4 ,-1 , 0
  4460.3     .16       0  4975.1     .07       0  5024.5     .16       0
  5538.6      .1       0
Bank Sta=4975.1,5024.5
XS Rating Curve= 0 ,0
Exp/Cntr=0.3,0.1

Type RM Length L Ch R = 1 ,84436   ,457,457,457
BEGIN DESCRIPTION:
SOUTH GRAPE CREEK 143.0
END DESCRIPTION:
XS GIS Cut Line= 4
      2765132.79     10013511.43      2765660.57     10013268.38
      2765764.73      10013053.1       2765806.4     10012608.66
#Sta/Elev= 30
  4325.9 1902.79  4365.2 1897.07  4420.2 1891.76  4486.3 1883.61  4541.3 1880.47
  4673.4 1870.37  4736.4 1868.97  4741.9 1866.53  4759.3 1861.26  4764.8 1857.24
  4772.5 1855.37  4787.8 1853.64  4902.6 1852.41  4955.3 1854.06  4977.9 1852.05
  5000.2 1846.94    5023 1851.84  5034.3 1854.13  5045.4 1854.79  5144.7 1852.75
  5205.7  1853.3  5326.3 1860.64  5344.1 1863.54  5349.1 1862.15  5366.4 1863.84
  5386.5 1864.14  5466.9 1875.76  5556.7 1885.21  5567.3 1887.92  5592.5 1892.22
#Mann= 4 ,-1 , 0
  4325.9     .16       0  4977.9     .07       0    5023     .16       0
  5592.5     .05       0
Bank Sta=4977.9,5023
XS Rating Curve= 0 ,0
Exp/Cntr=0.3,0.1

Type RM Length L Ch R = 1 ,83979   ,377,377,377
BEGIN DESCRIPTION:
SOUTH GRAPE CREEK 142.0
END DESCRIPTION:
XS GIS Cut Line= 3
       2766771.7     10014080.91      2765980.01     10013025.32
       2765993.9     10012560.02
#Sta/Elev= 30
  3813.8 1889.21  3992.9 1876.65    4072 1873.32  4078.3 1874.61  4092.9 1872.95
  4099.1 1874.24    4222 1868.84  4263.7 1869.55    4322 1865.89  4385.3 1865.81
  4485.3 1862.19  4528.3 1862.14  4542.9 1860.39  4592.9  1859.2  4799.1 1858.95
  4857.4 1856.66  4928.3 1856.71    4972 1849.04  4985.3  1845.6  4998.9 1844.16
  5035.3 1848.59  5049.1 1850.73  5092.9 1849.59  5249.5 1849.87    5305 1852.55
    5315 1854.44    5345 1865.68    5465 1900.54  5535.1 1912.54  5598.8 1918.99
#Mann= 4 ,-1 , 0
  3813.8     .16       0    4972     .07       0  5035.3     .16       0
  5598.8     .16       0
Bank Sta=4972,5035.3
XS Rating Curve= 0 ,0
Exp/Cntr=0.3,0.1

Type RM Length L Ch R = 1 ,83602   ,423,423,423
BEGIN DESCRIPTION:
SOUTH GRAPE CREEK 141.0
END DESCRIPTION:
XS GIS Cut Line= 2
      2766973.07     10013796.16      2766161.39      10012637.6
#Sta/Elev= 30
  3862.5 1882.91  3902.4 1881.34  3946.9 1875.06  3975.4 1875.65  4018.4 1871.09
    4075 1869.55  4104.7 1865.43  4134.1 1865.88    4191 1861.59  4247.7 1862.06
    4313 1858.96  4643.4 1850.54  4893.6 1849.15  4973.8 1846.12  4994.5 1839.58
  5009.6 1840.17  5015.7 1843.77  5024.4 1845.43  5030.5 1845.86  5081.1  1845.4
    5102 1848.47  5116.8 1853.99  5131.6  1885.2  5146.4 1895.89  5152.6  1896.9
  5167.4  1903.9  5188.3 1906.75  5203.1 1912.06  5274.6 1922.38  5277.1 1924.58
#Mann= 4 ,-1 , 0
  3862.5     .16       0  4973.8     .07       0  5030.5     .16       0
  5277.1     .16       0
Bank Sta=4973.8,5024.4
XS Rating Curve= 0 ,0
Exp/Cntr=0.3,0.1

Type RM Length L Ch R = 1 ,83179   ,664,664,664
BEGIN DESCRIPTION:
SOUTH GRAPE CREEK 140.0
END DESCRIPTION:
XS GIS Cut Line= 3
       2767334.2     10013719.79       2766681.4      10012803.1
      2766639.74     10012539.24
#Sta/Elev= 30
  3755.8 1891.64  3807.5 1887.96  3843.1 1882.32    3864 1882.42  3893.6 1877.98
  3922.8 1877.79  3971.9 1872.25  4015.3  1871.9  4050.9 1867.69  4086.6 1867.75
  4130.9 1862.88  4151.8 1863.39  4193.5    1859  4237.8 1858.02  4266.6 1855.35
  4309.1  1855.1  4459.1 1848.53    4604 1845.91  4825.5  1843.5  4927.9 1843.89
  4951.4 1844.03  4961.5 1842.14    4999 1835.48  5001.8 1834.98    5005 1835.48
  5012.1 1837.88 5017.27  1842.7    5083 1875.73  5133.6 1895.77  5148.3 1897.65
#Mann= 6 ,-1 , 0
  3755.8     .05       0  4459.1     .16       0    4604     .05       0
  4927.9      .1       0    4999     .07       0    5005      .1       0
Bank Sta=4961.5,5017.27
XS Rating Curve= 0 ,0
Exp/Cntr=0.3,0.1

Type RM Length L Ch R = 1 ,82515   ,374,374,374
BEGIN DESCRIPTION:
SOUTH GRAPE CREEK 139.0
END DESCRIPTION:
XS GIS Cut Line= 2
      2768000.84     10013289.21      2766843.46     10012138.75
#Sta/Elev= 30
  3962.1 1887.41    4003 1882.52  4066.6 1879.76    4201 1867.68  4334.7 1859.86
  4413.1 1858.25  4483.7 1853.91  4643.5 1848.54  4720.2 1845.47  4772.7 1843.49
  4918.6 1839.48  4964.7 1838.91  4978.8 1834.17    4997 1827.44  4999.8 1826.94
    5003 1827.44  5014.2 1833.86  5035.4 1839.03  5064.5 1837.67  5325.3 1838.06
    5372 1840.77  5438.4 1846.22  5445.5 1849.76  5452.6 1849.93  5480.9 1857.92
    5488 1862.24  5509.2 1868.44  5516.2 1873.19  5530.4 1878.11    5594 1897.06
#Mann= 11 ,-1 , 0
  3962.1      .1       0  4334.7     .05       0  4483.7      .1       0
  4643.5     .05       0  4720.2      .1       0  4772.7     .05       0
  4918.6      .1       0    4997     .07       0    5003      .1       0
  5064.5     .05       0    5372      .1       0
Bank Sta=4978.8,5014.2
XS Rating Curve= 0 ,0
Exp/Cntr=0.3,0.1

Type RM Length L Ch R = 1 ,82141   ,454,454,454
BEGIN DESCRIPTION:
SOUTH GRAPE CREEK 138.0
END DESCRIPTION:
XS GIS Cut Line= 3
      2768348.09     10012969.79      2767598.07     10012310.04
      2766868.91     10011962.83
#Sta/Elev= 30
  3845.6 1891.15  3866.6 1887.65  3977.5 1876.88  4047.7 1874.57  4183.4 1868.04
  4246.3 1862.51  4267.9  1863.2    4296 1860.74  4508.9 1848.44  4693.8 1843.21
  4821.1 1840.04  4865.7 1838.53    4894 1835.04    4977 1833.92  4984.8 1826.51
  4996.1 1823.86  4998.9 1823.36  5002.1 1823.86  5021.3 1829.91  5030.2 1834.81
  5116.2 1833.95  5245.6 1833.48  5397.9  1837.7  5432.9 1840.95  5472.7 1852.46
  5518.1 1872.04  5552.9 1889.99  5597.3 1906.77    5620 1911.15  5652.1 1911.81
#Mann= 12 ,-1 , 0
  3845.6      .1       0  3866.6     .16       0  4047.7     .05       0
  4183.4      .1       0  4246.3     .05       0    4296      .1       0
  4693.8     .05       0  4821.1      .1       0  4996.1     .07       0
  5002.1      .1       0  5116.2     .05       0  5432.9      .1       0
Bank Sta=4977,5030.2
XS Rating Curve= 0 ,0
Exp/Cntr=0.3,0.1

Type RM Length L Ch R = 1 ,81687   ,319,319,319
BEGIN DESCRIPTION:
SOUTH GRAPE CREEK 137.0
END DESCRIPTION:
XS GIS Cut Line= 3
      2768535.56     10012705.87      2767577.23     10011775.32
      2767049.45     10011733.66
#Sta/Elev= 30
  3775.6 1887.51  3867.1 1885.03  3944.8  1876.4  3990.8 1874.29  4032.9 1870.81
  4107.3 1864.35  4169.2 1862.41  4263.2 1859.17    4461 1840.49    4567 1837.44
  4659.1  1837.5  4814.7 1833.92  4868.1 1831.14  4963.1 1829.91  4977.3 1828.27
  4995.4 1821.47  4998.1 1820.97  5001.4 1821.47  5003.8 1822.09  5019.7  1829.5
  5031.5 1830.43  5120.2 1830.36  5195.3 1834.08  5220.5 1838.46  5280.7 1855.05
  5318.3 1862.17    5381 1873.81  5481.3 1882.55  5541.5  1894.1  5640.8 1898.08
#Mann= 11 ,-1 , 0
  3775.6     .16       0  3990.8     .05       0  4032.9      .1       0
  4169.2     .05       0  4263.2      .1       0  4868.1     .05       0
  4995.4    .035       0  5001.4     .05       0  5003.8      .1       0
  5031.5     .05       0  5318.3      .1       0
Bank Sta=4977.3,5019.7
XS Rating Curve= 0 ,0
Exp/Cntr=0.3,0.1

Type RM Length L Ch R = 1 ,81368   ,520,520,520
BEGIN DESCRIPTION:
SOUTH GRAPE CREEK 136.0
END DESCRIPTION:
XS GIS Cut Line= 3
      2768653.65     10012525.35       2767931.4     10011657.27
      2767174.43     10011150.31
#Sta/Elev= 30
    3729 1883.55  3778.3 1882.23  3883.2  1871.8  4016.8 1863.71  4045.9 1860.92
  4160.4 1856.64  4323.2  1839.3  4380.5 1835.43  4614.8 1829.58  4830.4 1828.56
  4970.1 1827.31  4984.8 1825.14  4996.8 1818.94  4999.5 1818.44  5002.8 1818.94
  5015.7  1822.7  5029.8  1825.9  5114.5 1826.48  5179.9 1832.19  5209.9 1838.78
    5273 1864.58    5288 1868.89    5309 1872.41  5369.4 1873.93  5390.5 1875.26
  5426.1 1875.94  5468.1 1883.86    5620 1887.95  5741.8 1888.81  5769.3 1888.91
#Mann= 10 ,-1 , 0
    3729     .16       0  3778.3     .05       0  4016.8      .1       0
  4830.4     .05       0  4996.8    .035       0  5002.8     .05       0
  5015.7      .1       0  5369.4     .16       0  5390.5      .1       0
  5741.8     .16       0
Bank Sta=4984.8,5029.8
XS Rating Curve= 0 ,0
Exp/Cntr=0.3,0.1

Type RM Length L Ch R = 1 ,80848   ,892,892,892
BEGIN DESCRIPTION:
SOUTH GRAPE CREEK 135.0
END DESCRIPTION:
XS GIS Cut Line= 3
      2768764.74     10012608.68       2768118.9     10011073.93
      2767362.69     10011094.75
#Sta/Elev= 30
  3574.4 1883.72  3753.1 1881.65  3775.1 1880.38  3824.7 1873.85  3858.1 1871.18
  3935.5 1867.55  3998.3 1862.45  4131.7 1857.35    4295 1839.85  4400.8  1832.2
  4630.7 1824.71  4948.2 1822.48  4971.9  1820.7  4998.1 1814.92  5000.8 1814.42
  5004.1 1814.92  5011.9 1816.41  5019.4 1824.63  5024.8 1822.89  5033.6 1828.58
  5048.6 1832.12  5129.4  1837.6  5240.3 1839.69    5420 1858.88  5556.1 1862.48
  5651.2 1867.87  5739.7 1872.43  5880.2 1883.77  5975.3 1885.11    5996 1885.55
#Mann= 13 ,-1 , 0
  3574.4      .1       0  3824.7     .05       0  3858.1      .1       0
  3998.3     .05       0  4131.7      .1       0  4998.1     .07       0
  5004.1      .1       0  5129.4     .16       0  5240.3      .1       0
  5556.1     .16       0  5651.2      .1       0  5739.7     .16       0
  5975.3      .1       0
Bank Sta=4948.2,5019.4
XS Rating Curve= 0 ,0
Exp/Cntr=0.3,0.1

Type RM Length L Ch R = 1 ,79956   ,638,638,638
BEGIN DESCRIPTION:
SOUTH GRAPE CREEK 134.0
END DESCRIPTION:
XS GIS Cut Line= 3
      2769584.16     10011810.02      2769077.23     10011087.82
      2767868.85     10010886.43
#Sta/Elev= 30
  3991.8 1855.64  4028.9 1853.78  4043.7  1855.2  4099.8 1855.65  4165.7 1851.06
  4243.8 1842.21  4280.5 1841.66  4375.1 1836.75  4609.9 1829.15  4689.5 1826.85
  4754.9 1823.17  4796.7 1818.38  4862.1 1813.46  4943.9 1811.77  4972.6 1810.51
  4986.9 1809.66  4989.6 1809.16  4992.9 1809.66  5014.8 1809.84  5035.1 1812.76
  5050.7 1815.85  5420.7 1819.73  5535.7 1822.69  5598.2 1826.11  5664.1 1826.93
  5714.4 1830.47  5740.9 1830.39  5785.7 1831.34  5963.1 1842.99  6099.2 1849.64
#Mann= 9 ,-1 , 0
  3991.8      .1       0  4099.8     .05       0  4375.1      .1       0
  4609.9     .05       0  4972.6      .1       0  4986.9     .07       0
  4992.9      .1       0  5535.7     .05       0  5740.9      .1       0
Bank Sta=4943.9,5035.1
XS Rating Curve= 0 ,0
Exp/Cntr=0.3,0.1

Type RM Length L Ch R = 1 ,79318   ,262,262,262
BEGIN DESCRIPTION:
SOUTH GRAPE CREEK 133.0
END DESCRIPTION:
XS GIS Cut Line= 3
      2769688.33     10011560.01      2769028.62     10010407.27
      2769042.48     10009617.16
#Sta/Elev= 30
  3786.2 1856.21  3863.4 1851.07  3878.2 1849.41    3894  1845.3  3921.4 1845.11
  3958.8 1841.03    4070 1835.13  4216.4 1824.89  4566.1  1819.1  4692.1 1812.29
  4737.3 1811.68  4764.7 1806.29  4807.9 1803.03  4876.5 1803.45  4957.1 1801.44
  4969.1 1797.48  4997.7 1794.47  5000.5 1793.97  5003.7 1794.47  5022.3 1799.97
  5108.6 1805.94  5217.9  1810.5  5247.9 1816.19  5292.5 1828.43  5386.7 1851.71
  5475.3 1867.69    5588 1882.44    5688 1890.78    5828  1899.4  5904.6 1908.54
#Mann= 6 ,-1 , 0
  3786.2     .05       0  3863.4      .1       0  4997.7     .07       0
  5003.7      .1       0  5292.5     .16       0  5475.3      .1       0
Bank Sta=4957.1,5022.3
XS Rating Curve= 0 ,0
Exp/Cntr=0.3,0.1

Type RM Length L Ch R = 1 ,79056   ,370,370,370
BEGIN DESCRIPTION:
SOUTH GRAPE CREEK 132.0
END DESCRIPTION:
XS GIS Cut Line= 3
      2769736.95     10011268.37      2769355.01     10010469.77
      2769091.22     10010018.55
#Sta/Elev= 30
  3940.1 1835.02  4045.7 1829.74  4062.8 1826.93  4078.3 1828.22  4153.5 1822.18
  4198.9 1822.54    4311 1818.22  4333.2 1819.41  4385.8 1816.47  4482.1 1815.87
  4521.6 1813.46  4731.5 1809.51  4754.1 1803.97  4782.4 1801.04  4891.9 1798.68
  4959.7 1799.13  5000.5 1792.99  5003.3 1792.49  5006.5 1792.99    5025 1798.84
  5094.6 1803.61  5156.7  1816.3  5185.3  1825.9  5191.4 1830.21    5244 1852.69
  5265.5 1857.22  5281.2 1863.76  5302.7 1869.44  5345.7 1874.45    5348 1876.12
#Mann= 4 ,-1 , 0
  3940.1      .1       0  5000.5     .07       0  5006.5      .1       0
  5094.6     .16       0
Bank Sta=4959.7,5025
XS Rating Curve= 0 ,0
Exp/Cntr=0.3,0.1

Type RM Length L Ch R = 1 ,78686   ,403,403,403
BEGIN DESCRIPTION:
SOUTH GRAPE CREEK 131.0
END DESCRIPTION:
XS GIS Cut Line= 2
      2769799.46     10011171.16      2769542.52     10009948.97
#Sta/Elev= 30
  4084.5 1828.93  4210.2 1822.59  4327.1 1818.79    4368 1818.94  4419.1 1816.11
  4480.4 1816.21  4664.3 1810.59  4715.4  1807.1  4776.7 1806.85  4793.1  1803.8
  4858.5 1798.95  4919.8 1799.48  4981.1 1797.17  4992.5 1791.68  4998.5 1791.17
  5001.3 1790.67  5004.5 1791.17  5037.2 1796.12  5062.9  1796.7  5099.6 1801.94
  5186.8 1806.01  5216.1 1811.26  5226.4 1814.17  5231.5 1817.75  5236.6  1818.5
  5276.3 1837.33  5281.4  1838.5  5287.7 1843.68  5326.1 1862.22  5333.4 1863.23
#Mann= 4 ,-1 , 0
  4084.5      .1       0  4998.5     .07       0  5004.5      .1       0
  5099.6     .16       0
Bank Sta=4981.1,5037.2
XS Rating Curve= 0 ,0
Exp/Cntr=0.3,0.1

Type RM Length L Ch R = 1 ,78283   ,469,469,469
BEGIN DESCRIPTION:
SOUTH GRAPE CREEK 130.0
END DESCRIPTION:
XS GIS Cut Line= 3
      2769917.51     10011310.05      2770035.57     10010421.16
      2769924.46     10009789.25
#Sta/Elev= 30
  3846.2 1834.58  4003.7 1825.21  4179.4 1819.91  4688.4  1803.9  4731.1 1803.31
  4780.9 1797.58  4809.5 1796.36  4953.5  1796.1  4979.5 1790.98  4982.2 1790.48
  4985.5 1790.98  5041.8 1792.07  5046.9 1792.62    5055  1797.1    5061 1799.47
  5065.2 1801.13  5106.2 1803.84  5136.3 1811.05  5155.4 1819.43  5160.5 1819.68
  5214.7 1848.09  5219.8 1848.24  5237.8 1856.06    5274 1867.09  5285.4 1868.26
  5308.9 1868.57  5328.3 1865.65  5333.4 1867.24  5369.8 1859.72  5384.5 1858.18
#Mann= 8 ,-1 , 0
  3846.2     .05       0  4003.7      .1       0  4179.4     .05       0
  4688.4      .1       0  4979.5     .07       0  4985.5      .1       0
    5061     .16       0  5285.4      .1       0
Bank Sta=4953.5,5055
XS Rating Curve= 0 ,0
Exp/Cntr=0.3,0.1

Type RM Length L Ch R = 1 ,77814   ,540,540,540
BEGIN DESCRIPTION:
SOUTH GRAPE CREEK 129.0
END DESCRIPTION:
XS GIS Cut Line= 3
      2770348.06     10011442.03      2770473.07     10009879.49
      2770251.19     10009317.87
#Sta/Elev= 30
  3677.3  1832.6  3712.2 1830.57  3747.9 1829.35  3846.1 1820.69  3952.7 1816.25
  4042.3 1812.88  4121.6 1810.85  4157.1 1807.87  4177.2 1809.72  4448.1 1802.77
  4623.2 1800.56  4708.9 1796.46  4889.5 1795.74  4949.7 1792.98  4979.8 1787.69
  4998.9 1786.65  5001.7 1786.15  5004.9 1786.65  5039.9 1793.77  5119.8 1802.83
  5272.9 1807.64  5328.5 1809.23  5352.9 1814.38    5407 1836.76  5461.1 1852.58
  5531.7 1857.61  5593.6  1865.6  5707.2 1872.59  5767.1 1881.21  5848.7 1884.71
#Mann= 8 ,-1 , 0
  3677.3     .05       0  3712.2      .1       0  3952.7     .05       0
  4042.3      .1       0  4998.9     .07       0  5004.9      .1       0
  5272.9     .16       0  5531.7      .1       0
Bank Sta=4949.7,5039.9
XS Rating Curve= 0 ,0
Exp/Cntr=0.3,0.1

Type RM Length L Ch R = 1 ,77274   ,482,482,482
BEGIN DESCRIPTION:
SOUTH GRAPE CREEK 128.0
END DESCRIPTION:
XS GIS Cut Line= 3
      2770528.62      10011490.6      2770820.29      10010428.1
      2771444.38      10009762.4
#Sta/Elev= 30
  3799.7 1833.05  3816.1  1832.3  3996.1 1821.29  4118.6 1813.55  4329.6 1805.29
  4372.2 1803.53  4571.3 1796.37  4960.1 1790.09  4999.5  1784.8  5002.3  1784.3
  5005.5  1784.8  5034.5 1788.55  5044.6 1789.29  5129.6  1796.9  5292.2 1800.04
  5313.7 1802.02  5338.8 1808.87  5462.2 1849.31  5539.9 1866.72    5639 1873.64
  5674.7 1872.39  5681.5 1874.44  5709.7 1871.26  5730.9 1873.57  5738.2 1871.72
    5745 1873.71  5752.3 1871.92  5759.2 1873.75  5794.8 1872.26    5814 1875.28
#Mann= 11 ,-1 , 0
  3799.7      .1       0  3816.1     .05       0  3996.1      .1       0
  4118.6     .05       0  4329.6      .1       0  4372.2     .05       0
  4999.5    .035       0  5005.5     .05       0  5034.5      .1       0
  5338.8     .16       0  5709.7      .1       0
Bank Sta=4960.1,5044.6
XS Rating Curve= 0 ,0
Exp/Cntr=0.3,0.1

Type RM Length L Ch R = 1 ,76792   ,261,261,261
BEGIN DESCRIPTION:
SOUTH GRAPE CREEK 127.0
END DESCRIPTION:
XS GIS Cut Line= 2
      2770889.72     10011421.17      2771507.42     10010158.02
#Sta/Elev= 30
  4081.7 1823.27  4113.7 1820.29  4137.9 1820.46  4167.9 1816.48  4205.5 1816.36
  4234.7 1812.66  4274.2 1811.84  4340.5 1807.42  4379.4 1807.43  4617.6 1797.16
  4813.4 1791.46  4864.5 1790.46  4886.4 1787.94  4947.1  1786.5  4971.7 1785.07
    4996 1784.27  4998.7 1783.77    5002 1784.27  5021.5 1784.34  5036.2 1787.38
  5118.2 1792.09  5186.2 1793.16  5224.1 1795.63  5246.6 1800.47  5303.3  1824.9
    5359  1844.4  5370.3 1850.06  5403.5 1859.46  5415.4 1864.77  5487.8 1884.97
#Mann= 11 ,-1 , 0
  4081.7      .1       0  4113.7     .05       0  4274.2      .1       0
  4617.6     .05       0  4813.4      .1       0  4864.5     .05       0
  4971.7     .16       0    4996     .07       0    5002     .16       0
  5118.2      .1       0  5186.2     .16       0
Bank Sta=4947.1,5036.2
XS Rating Curve= 0 ,0
Exp/Cntr=0.3,0.1

Type RM Length L Ch R = 1 ,76531   ,512,512,512
BEGIN DESCRIPTION:
SOUTH GRAPE CREEK 126.0
END DESCRIPTION:
XS GIS Cut Line= 2
      2771209.18     10011428.09      2771722.81     10010248.13
#Sta/Elev= 30
  4252.9 1819.32  4254.7 1819.32  4395.3 1810.97  4432.2 1810.75  4475.8  1807.1
  4530.3 1805.96  4595.7 1801.33  4908.9 1790.81  4963.1 1787.57  4977.5 1784.33
    5007 1784.21  5009.8 1783.71    5013 1784.21  5014.2 1784.32    5032  1787.4
  5091.2 1786.71    5167 1788.52  5242.7 1793.43  5266.2 1798.68  5289.6 1808.54
  5341.9 1826.43  5365.4 1837.15  5388.8  1845.2  5394.2 1845.83  5412.2 1853.31
  5435.5 1859.37  5441.1 1862.44  5464.5 1868.96  5493.4 1873.33  5539.8 1884.63
#Mann= 7 ,-1 , 0
  4252.9      .1       0  4254.7     .05       0  4395.3      .1       0
  4908.9     .05       0    5007    .035       0    5013     .05       0
  5014.2     .16       0
Bank Sta=4963.1,5032
XS Rating Curve= 0 ,0
Exp/Cntr=0.3,0.1

Type RM Length L Ch R = 1 ,76019   ,299,299,299
BEGIN DESCRIPTION:
SOUTH GRAPE CREEK 125.0
END DESCRIPTION:
XS GIS Cut Line= 3
      2771646.69     10011594.74       2771993.9     10010726.71
      2771959.18     10010310.05
#Sta/Elev= 30
  4205.8 1822.42  4324.7 1812.49  4346.9 1812.58  4368.4 1809.55  4409.3 1807.41
  4444.3 1803.71  4486.9 1802.55  4522.4 1799.75  4562.3 1799.06  4654.4 1793.69
  4863.9 1787.99  4899.4 1784.35  4977.5 1785.14  4982.9 1784.44  5001.7 1784.94
  5006.8 1783.83  5025.4 1784.77  5031.3    1785  5079.3 1784.63  5109.4 1786.63
  5267.7 1784.83  5304.2  1787.7  5354.4 1788.81  5388.1 1791.09  5404.6 1793.24
  5434.7 1801.16  5508.6 1833.48    5515 1837.67  5554.4 1853.08  5558.8 1853.08
#Mann= 4 ,-1 , 0
  4205.8      .1       0  4324.7     .16       0  4982.9     .07       0
  5025.4     .16       0
Bank Sta=4977.5,5031.3
XS Rating Curve= 0 ,0
Exp/Cntr=0.3,0.1

Type RM Length L Ch R = 1 ,75720   ,124,124,124
BEGIN DESCRIPTION:
SOUTH GRAPE CREEK 124.0
END DESCRIPTION:
XS GIS Cut Line= 4
      2771939.22     10011615.59      2772217.86     10010941.12
      2772251.71     10010826.54      2772066.83     10010271.88
#Sta/Elev= 30
  4335.2 1817.91  4421.6 1809.19  4467.1 1806.88  4488.7 1803.68  4521.2 1802.74
    4552  1799.5  4586.8 1799.88  4618.5 1796.33    4765 1790.09  4842.1 1788.78
  4866.1 1786.33  4871.5 1784.64  4895.4 1785.01  4942.9  1783.4    5008 1784.09
  5188.6 1784.03  5282.3 1785.92  5535.3 1784.69    5618 1793.96  5640.7 1799.23
  5654.9 1804.09  5661.7 1808.11  5686.5 1818.65  5693.4  1823.2  5712.8 1832.57
  5718.1 1833.55  5744.5 1846.23  5749.7    1847  5765.5 1854.32  5769.1 1854.32
#Mann= 4 ,-1 , 0
  4335.2      .1       0  4895.4     .07       0    5008      .1       0
  5769.1     .16       0
Bank Sta=4895.4,5008
XS Rating Curve= 0 ,0
Exp/Cntr=0.3,0.1

Type RM Length L Ch R = 1 ,75596   ,152,152,152
BEGIN DESCRIPTION:
Mapping XS c15b15bf
END DESCRIPTION:
XS GIS Cut Line= 4
      2772025.16     10011620.79      2772327.23     10011006.22
      2772332.44     10010883.83      2772144.95     10010258.85
#Sta/Elev= 30
  4367.5 1816.52  4451.1 1807.77  4479.1    1807  4509.1 1802.94  4642.8 1794.18
  4703.9 1791.61  4799.4 1790.03  4844.3 1791.48  4861.2 1793.47  4866.8 1792.59
  4883.7 1795.41  4889.3 1794.31  4906.2 1796.71  4973.6 1798.27  5017.1 1797.04
  5041.1 1798.77  5046.6 1797.37  5124.9 1795.93  5195.8 1790.31  5216.7 1787.14
  5279.8 1782.79  5289.7 1784.21  5384.5 1785.59  5582.1    1784    5676 1789.61
  5686.5 1791.44  5730.8 1808.49  5796.9 1842.33  5822.2 1852.52  5827.3 1852.52
#Mann= 4 ,-1 , 0
  4367.5      .1       0  4973.6     .05       0  5041.1      .1       0
  5827.3     .16       0
#XS Ineff= 2 , 0
       0 4951.37 1797.97  5064.9       0 1798.12
Permanent Ineff=
       T       T
Bank Sta=4973.6,5041.1
XS Rating Curve= 0 ,0
Exp/Cntr=0.3,0.1

Type RM Length L Ch R = 1 ,75444   ,447,447,447
BEGIN DESCRIPTION:
SOUTH GRAPE CREEK 123.0
END DESCRIPTION:
XS GIS Cut Line= 4
      2772163.17     10011685.91       2772496.5     10010998.41
      2772488.69     10010839.56      2772272.99     10010244.44
#Sta/Elev= 30
    4343 1821.02  4445.4 1808.54  4489.9 1806.42  4522.4 1802.89  4550.5  1802.4
  4567.5 1799.67  4708.5 1791.94  4804.4 1790.24  4917.2  1785.9  4967.9 1777.81
  4990.5 1772.39  5000.9 1771.87  5023.3  1777.1  5121.7 1778.62  5172.9 1782.03
  5201.8 1786.15  5241.9 1783.58  5346.7 1782.66  5474.4 1784.87  5636.4 1784.13
    5687 1787.83  5761.6 1789.98  5784.2 1794.02  5804.1 1801.59  5809.6 1805.71
  5814.9 1806.66  5840.2 1817.47  5865.5 1831.28  5889.2 1840.51  5899.1 1845.87
#Mann= 5 ,-1 , 0
    4343      .1       0  4967.9     .05       0  4967.9     .07       0
  5023.3      .1       0  5899.1     .16       0
Bank Sta=4967.9,5023.3
XS Rating Curve= 0 ,0
Exp/Cntr=0.3,0.1

Type RM Length L Ch R = 1 ,74997   ,664,664,664
BEGIN DESCRIPTION:
SOUTH GRAPE CREEK 122.0
END DESCRIPTION:
XS GIS Cut Line= 3
      2772540.75     10011787.51      2772926.19     10011131.22
      2772915.78     10010204.19
#Sta/Elev= 30
  4393.1 1815.87    4438 1814.89  4501.6  1809.3  4555.2 1805.26  4629.4 1802.12
  4789.7 1792.47  4869.8 1788.61  4934.2 1787.44  4955.6 1785.17  4971.3 1781.15
  4977.3 1776.46    4987 1771.53  5000.3 1769.55  5014.3 1771.27  5029.9 1775.89
  5051.4 1776.74  5067.1 1774.71  5088.5    1774  5147.2 1775.63  5221.7 1774.46
  5301.7 1776.26  5341.7 1775.57  5471.7 1779.59  5781.7 1780.55  5891.7 1784.36
  5911.7 1785.77  5931.7 1789.79  5986.7 1808.64  6031.8 1825.41  6081.3 1838.98
#Mann= 6 ,-1 , 0
  4393.1     .05       0  4501.6     .16       0  4977.3     .07       0
  5014.3     .16       0  5931.7      .1       0  5986.7     .16       0
Bank Sta=4977.3,5029.9
XS Rating Curve= 0 ,0
Exp/Cntr=0.3,0.1

Type RM Length L Ch R = 1 ,74333   ,370,370,370
BEGIN DESCRIPTION:
SOUTH GRAPE CREEK 121.0
END DESCRIPTION:
XS GIS Cut Line= 3
      2772780.34      10011912.5      2773322.02     10010995.81
      2773124.11      10010303.1
#Sta/Elev= 30
  3784.5 1812.19  3811.2 1812.37  3861.8  1808.8  3885.4 1806.17  3906.8 1807.13
  3949.7 1803.19  4058.8 1798.02  4242.3 1791.61  4482.2 1787.68  4636.3 1781.87
  4657.8 1779.46  4861.8 1775.84  4934.6 1771.66  4965.8 1770.25    4994 1765.58
  4996.8 1765.08  5024.5 1767.06  5029.7 1769.48    5049 1772.06  5090.6 1775.49
  5184.2 1778.62  5315.7 1777.11  5402.6 1779.36  5461.2 1782.33  5500.3 1786.28
  5527.4 1795.49  5534.1 1799.65  5539.3 1798.87  5564.8 1810.25  5569.7 1811.28
#Mann= 8 ,-1 , 0
  3784.5     .05       0  3861.8      .1       0  4058.8     .16       0
    4994     .07       0  5024.5     .16       0  5402.6     .05       0
  5461.2      .1       0  5564.8     .16       0
#XS Ineff= 2 , 0
                         5195.02            1779
Permanent Ineff=
       T       T
Bank Sta=4934.6,5049
XS Rating Curve= 0 ,0
Exp/Cntr=0.3,0.1

Type RM Length L Ch R = 1 ,73963   ,402,402,402
BEGIN DESCRIPTION:
SOUTH GRAPE CREEK 120.0
END DESCRIPTION:
XS GIS Cut Line= 3
      2773339.51      10012119.8      2773629.32     10010792.68
      2773535.75     10010267.65
#Sta/Elev= 30
  3547.4 1799.06  3625.3 1797.07  3809.5 1792.14  3890.2 1792.52  4179.2 1786.37
    4218 1787.03  4687.8 1774.61  4878.7 1772.38  4902.7 1768.25  4945.4 1769.51
    4986  1768.3  4995.7 1765.15  4998.4 1764.65  5001.7 1765.15  5026.6 1767.87
  5111.5 1769.82  5224.4 1778.36  5260.2 1783.15  5270.4 1786.11  5278.3 1790.37
  5283.4  1790.7  5290.7 1795.21  5331.3 1813.64  5337.3 1817.67  5342.3 1818.34
  5391.2 1837.33  5396.2 1837.38  5402.4 1841.06  5432.9 1851.17  5439.1 1854.35
#Mann= 4 ,-1 , 0
  3547.4     .05       0  3625.3     .16       0  4995.7     .07       0
  5001.7     .16       0
Bank Sta=4986,5026.6
XS Rating Curve= 0 ,0
Exp/Cntr=0.3,0.1

Type RM Length L Ch R = 1 ,73561   ,776,776,776
BEGIN DESCRIPTION:
SOUTH GRAPE CREEK 119.0
END DESCRIPTION:
XS GIS Cut Line= 3
      2773655.35      10011839.6      2773967.86     10010693.72
      2773978.26     10010288.08
#Sta/Elev= 30
  3673.4 1787.45    3863 1784.61  3878.5 1784.54  3938.6 1783.63  4021.5  1781.8
    4063 1783.23  4135.5 1780.13  4269.7 1778.39  4394.7  1773.3    4405 1774.41
  4508.7 1771.86  4633.1 1770.07    4716 1770.72    4845 1768.05  4891.1 1768.88
  4931.1 1765.34  4961.1 1765.78  5010.9  1762.3  5031.2 1765.69  5041.2 1768.44
    5078 1791.54    5083 1791.29  5091.2 1794.37  5101.2 1795.54  5111.2 1799.31
  5151.2 1820.47  5161.2 1830.15  5171.2 1834.43  5221.2 1839.58  5266.9 1839.33
#Mann= 6 ,-1 , 0
  3673.4     .05       0    3863      .1       0  3878.5     .05       0
  3938.6     .16       0  4961.1     .07       0  5031.2     .16       0
Bank Sta=4961.1,5031.2
XS Rating Curve= 0 ,0
Exp/Cntr=0.3,0.1

Type RM Length L Ch R = 1 ,72785   ,413,413,413
XS GIS Cut Line= 5
      2773686.07     10012056.68      2774513.89     10010948.03
      2774511.45     10010852.79      2774411.33     10010669.64
      2774103.64     10010344.86
#Sta/Elev= 30
  3774.6 1787.57  3785.7 1787.39  3956.7 1783.49  4165.2 1781.81  4171.4  1780.5
  4464.7 1775.73    4507 1773.59  4536.2 1774.53  4627.9 1771.96    4728 1771.68
  4764.2 1769.97  4786.4 1765.93    4828 1761.98  4971.9 1760.35  4992.5 1753.38
  5036.5 1757.26  5042.8 1760.68  5051.1 1761.19  5057.4 1766.47  5086.6 1768.46
  5162.9 1767.69  5416.9 1770.51  5532.1  1774.1  5588.7 1779.42  5652.2 1788.36
  5673.7 1793.14    5702 1802.35  5793.8  1821.4  5822.1 1828.88  5909.6 1835.26
#Mann= 5 ,-1 , 0
  3774.6     .05       0  3785.7     .16       0  4971.9     .07       0
  5057.4     .16       0  5909.6      .1       0
Bank Sta=4971.9,5042.8
XS Rating Curve= 0 ,0
Exp/Cntr=0.3,0.1

Type RM Length L Ch R = 1 ,72372   ,227,227,227
BEGIN DESCRIPTION:
SOUTH GRAPE CREEK 117.0
END DESCRIPTION:
XS GIS Cut Line= 5
      2773819.27       10012169.      2774475.31     10011755.94
      2774627.16     10011315.56      2774587.68     10010653.48
      2774187.19     10009947.73
#Sta/Elev= 30
  3899.7 1785.17  3981.5 1784.64  4048.4 1780.05  4148.5 1777.36  4206.2 1777.62
  4236.8  1775.3  4519.4 1769.19  4598.3 1769.95  4673.9 1766.54    4915 1766.31
  4962.9 1763.96  4972.1 1762.23  4977.4 1757.59    4984 1753.08  4999.8 1750.82
  5039.8 1755.79  5058.1 1756.42  5121.6 1757.86  5139.1 1761.45  5162.6 1762.46
  5292.9 1761.68  5312.9 1764.27  5870.2 1771.48  6148.7 1780.59  6360.5 1796.66
  6419.7 1798.17  6462.9 1803.73  6581.2 1814.53  6602.8  1820.7  6615.5 1822.67
#Mann= 3 ,-1 , 0
  3899.7     .16       0  4972.1     .07       0  5058.1     .16       0
Bank Sta=4977.4,5058.1
XS Rating Curve= 0 ,0
Exp/Cntr=0.3,0.1

Type RM Length L Ch R = 1 ,72145   ,282,282,282
XS GIS Cut Line= 6
      2774049.91     10012159.27      2774697.04     10011746.57
       2774816.7     10011380.27      2774994.97     10010882.09
      2775024.28     10010132.39       2775214.1     10009730.83
#Sta/Elev= 30
  4005.4 1776.84    4008 1776.91  4247.5 1770.23  4638.5 1764.39  4965.3 1764.78
  4983.9    1751  4996.6 1749.94  5015.8 1752.66  5079.6 1754.93    5102 1751.23
  5165.2 1756.88  5210.5  1754.5  5259.7 1757.52  5384.5 1764.56  5420.6 1766.34
  5502.3 1764.56  5507.6 1766.75  5533.1 1765.63  5538.4 1767.94  5681.6 1770.93
  5687.4  1768.4  5755.8  1771.7  5986.2 1772.02  6046.3 1775.54  6386.4 1780.88
  6408.8 1783.87  6649.2 1793.43  6711.9 1793.69    6854 1802.99  6881.9  1805.6
#Mann= 5 ,-1 , 0
  4005.4     .05       0    4008     .16       0  5165.2     .07       0
  5259.7     .16       0    6854     .05       0
Bank Sta=4965.3,5384.5
XS Rating Curve= 0 ,0
Exp/Cntr=0.3,0.1

Type RM Length L Ch R = 1 ,71863   ,437,437,437
XS GIS Cut Line= 4
      2774092.61     10012196.34      2774870.13     10011762.02
      2775377.33      10010884.3      2776074.64     10010584.15
#Sta/Elev= 30
    3773 1774.33    4052 1767.29  4382.2 1762.98    4501 1762.94  4550.1 1764.88
  4711.9 1762.47  4904.2 1762.94  4925.8 1758.91  4947.3 1753.13  4993.6 1748.03
  4996.3 1747.53    5012 1748.06  5049.3 1753.93  5135.4  1759.3  5296.8 1767.17
  5547.4 1772.93  5792.7 1787.67  5839.8 1794.78  5868.8 1794.72  5892.3  1801.5
  5997.3 1815.99  6020.9 1820.57  6044.4 1828.31  6135.8 1842.31    6173 1848.75
  6196.5 1855.18    6220 1858.18    6325 1862.83  6372.1 1867.92  6436.5 1869.44
#Mann= 4 ,-1 , 0
    3773     .16       0  4993.6     .07       0  5135.4     .16       0
  6135.8     .16       0
Bank Sta=4925.8,5135.4
XS Rating Curve= 0 ,0
Exp/Cntr=0.3,0.1

Type RM Length L Ch R = 1 ,71426   ,369,369,369
BEGIN DESCRIPTION:
SOUTH GRAPE CREEK 115.0
END DESCRIPTION:
XS GIS Cut Line= 3
      2774311.64      10012188.5       2775368.9     10011599.97
       2775753.4     10011168.72
#Sta/Elev= 30
  3635.7 1767.49  3723.6 1766.88  3798.9 1763.22  3982.9 1761.46  4113.3 1763.17
  4226.5 1761.42  4387.4 1764.11  4578.6 1758.75  4719.3 1757.47  4845.7 1753.59
  4870.9  1751.2  4913.5 1752.34  4934.5 1750.99    4942 1747.65  4962.9  1745.3
  4984.6 1747.17  5005.3 1744.45  5019.7 1747.77 5023.86    1752  5033.9 1759.52
  5041.4 1768.14  5048.1 1771.85  5055.1 1779.63  5062.4 1783.37  5076.6 1785.65
  5168.5 1790.63  5225.4  1796.6  5282.2 1799.06  5331.6 1803.79  5423.5 1808.25
#Mann= 4 ,-1 , 0
  3635.7     .16       0  4934.5     .07       0  5019.7     .16       0
  5423.5      .1       0
Bank Sta=4934.5,5023.86
XS Rating Curve= 0 ,0
Exp/Cntr=0.3,0.1

Type RM Length L Ch R = 1 ,71057   ,502,502,502
BEGIN DESCRIPTION:
SOUTH GRAPE CREEK 114.0
END DESCRIPTION:
XS GIS Cut Line= 3
       2774478.4     10012230.88      2775672.85     10011772.55
       2776221.5     10011341.96
#Sta/Elev= 30
  3610.1 1763.17  3610.5 1763.17  3749.4 1760.78  3839.9 1762.43  3877.9 1759.78
  4392.1 1762.69  4445.6 1761.42  4520.6 1754.34  4870.5 1755.92  4892.9 1755.24
  4913.8 1749.69  4942.7 1752.51  4957.1 1749.56  4977.9  1741.2  4989.4 1740.54
  4992.1 1740.04  4995.4 1740.54    5071 1749.27  5135.2 1760.56    5156 1766.68
  5163.6 1765.96  5176.8 1770.29  5184.9 1770.31  5234.6  1783.4  5334.1 1792.76
  5377.4 1802.33  5427.2 1803.42  5555.5 1812.05  5557.7 1812.43  5586.9 1813.29
#Mann= 7 ,-1 , 0
  3610.1     .05       0  3610.5      .1       0  3877.9     .16       0
  4989.4     .07       0  4995.4     .16       0  5555.5      .1       0
  5557.7     .16       0
#XS Ineff= 2 , 0
         4850.62 1755.97
Permanent Ineff=
       T       T
Bank Sta=4957.1,5071
XS Rating Curve= 0 ,0
Exp/Cntr=0.3,0.1

Type RM Length L Ch R = 1 ,70555   ,1080,1080,1080
BEGIN DESCRIPTION:
SOUTH GRAPE CREEK 113.0
END DESCRIPTION:
XS GIS Cut Line= 3
      2774306.36     10012329.15      2776202.23     10012094.77
      2776639.72     10011855.19
#Sta/Elev= 30
  3324.9  1767.4  3411.2 1766.59  3437.9 1764.41  3609.2 1760.39  3679.7 1761.53
    3720 1756.28  3800.6 1755.53  3871.1 1759.08  4145.8 1761.43  4307.9 1755.75
  4374.9 1749.61  4425.3 1748.13  4495.9 1749.89  4606.7 1748.19  4828.4 1750.31
  4939.2 1747.12  4996.7 1738.76  4999.4 1738.26  5002.7 1738.76  5029.9 1742.33
  5037.4 1748.46  5042.4 1747.13  5060.1 1767.23  5070.2 1775.04  5080.3 1778.92
  5118.5 1784.39  5123.5 1783.04  5211.3 1790.47  5595.8 1805.61    5734 1812.86
#Mann= 5 ,-1 , 0
  3324.9     .05       0  3437.9     .16       0  4996.7     .07       0
  5002.7     .16       0    5734     .16       0
#XS Ineff= 2 , 0
         4142.74 1761.79
Permanent Ineff=
       T       T
Bank Sta=4939.2,5037.4
XS Rating Curve= 0 ,0
Exp/Cntr=0.3,0.1
