HEC-RAS study SOUTH GRAPE CREEK.prj: SOUTH GRAPE CREEK Base Level Engineering

--- SOUTH GRAPE CREEK.g01 (geometry) --- (continued)

Type RM Length L Ch R = 1 ,47401   ,832,832,832
BEGIN DESCRIPTION:
SOUTH GRAPE CREEK 72.0
END DESCRIPTION:
XS GIS Cut Line= 4
      2784327.58     10027138.31      2784718.21     10026471.63
      2785134.87     10026247.67       2785774.2     10025509.59
#Sta/Elev= 30
  4045.4 1664.66  4164.9 1659.62  4269.9 1649.25  4334.3 1632.25  4355.8 1622.12
  4386.8 1627.61  4531.7 1633.26  4596.2 1627.64  4782.1  1630.6  4857.6 1629.86
  4911.8 1627.09  4990.8 1616.67  4993.5 1616.17  4996.8 1616.67  5059.5 1622.24
  5075.8 1626.59  5119.6 1631.48  5201.6  1632.6  5242.3 1635.69  5360.6 1638.82
  5374.9 1643.04  5384.7 1642.84  5430.8 1641.17  5599.7 1645.04  5635.6 1645.56
  5740.6 1646.37    5983 1649.22  6054.9 1648.98  6167.7 1653.39  6267.6 1656.83
#Mann= 13 ,-1 , 0
  4045.4      .1       0  4164.9     .16       0  4782.1      .1       0
  4857.6     .16       0  4990.8     .07       0  4996.8     .16       0
  5242.3     .05       0  5384.7      .1       0  5599.7     .05       0
  5635.6      .1       0  5740.6     .05       0    5983      .1       0
  6167.7     .05       0
Bank Sta=4911.8,5075.8
XS Rating Curve= 0 ,0
Exp/Cntr=0.3,0.1

Type RM Length L Ch R = 1 ,46569   ,534,534,534
BEGIN DESCRIPTION:
SOUTH GRAPE CREEK 71.0
END DESCRIPTION:
XS GIS Cut Line= 3
      2784588.02     10027580.98      2785145.29     10026919.55
      2785739.02       10025680.
#Sta/Elev= 30
  4438.8 1673.63  4519.8 1669.96  4629.8 1664.95    4754 1659.44  4799.5 1656.95
  4878.1 1647.98  4933.5 1641.52  4962.1 1624.66  4969.9 1620.11    5002 1611.73
  5004.7 1611.23    5008 1611.73  5054.4 1617.81  5132.5 1623.94  5136.5 1623.75
  5161.1 1622.68  5203.9 1626.82    5282 1629.14  5504.1 1628.16  5633.7 1631.43
  5775.8 1632.73    6004  1640.8  6112.8 1645.23  6186.1 1643.87  6225.2 1647.05
  6287.6 1645.54  6366.7 1644.68  6638.9 1649.53  6666.8 1651.87  6678.1 1649.97
#Mann= 14 ,-1 , 0
  4438.8      .1       0  4519.8     .16       0  4629.8      .1       0
    4754     .16       0  4878.1      .1       0    5002     .07       0
    5008      .1       0  5136.5     .16       0  5504.1      .1       0
  5633.7     .16       0    6004     .05       0  6112.8      .1       0
  6287.6     .05       0  6638.9      .1       0
Bank Sta=4962.1,5132.5
XS Rating Curve= 0 ,0
Exp/Cntr=0.3,0.1

Type RM Length L Ch R = 1 ,46035   ,728,728,728
BEGIN DESCRIPTION:
SOUTH GRAPE CREEK 70.0
END DESCRIPTION:
XS GIS Cut Line= 3
       2785030.7     10028039.35      2785561.96     10027122.67
      2785905.63     10025508.44
#Sta/Elev= 30
  4236.6 1665.66    4348 1661.91  4573.6 1655.67  4791.5 1647.34  4902.6 1642.62
  4941.2 1636.68  4962.8 1628.76  4978.5 1617.12    4997 1610.37  4999.8 1609.87
    5003 1610.37    5008 1611.17  5080.4 1618.02  5096.1 1615.34  5133.1 1616.99
  5160.7 1615.61  5209.3 1623.72    5594  1624.1  5941.9 1632.01  6019.5 1633.75
  6122.1 1638.32  6194.7 1641.94  6238.2 1641.46    6297 1640.06  6367.3 1642.04
  6562.8 1645.96  6763.6 1653.05  6808.8 1654.71  6914.1 1657.78  6946.5 1659.36
#Mann= 17 ,-1 , 0
  4236.6     .16       0    4348      .1       0  4573.6     .16       0
  4791.5      .1       0  4902.6     .16       0    4997     .07       0
    5003     .16       0    5008      .1       0  5209.3     .16       0
  5941.9      .1       0  6019.5     .16       0  6122.1     .05       0
  6238.2      .1       0  6367.3     .05       0  6763.6      .1       0
  6808.8     .05       0  6914.1      .1       0
Bank Sta=4978.5,5080.4
XS Rating Curve= 0 ,0
Exp/Cntr=0.3,0.1

Type RM Length L Ch R = 1 ,45307   ,469,469,469
BEGIN DESCRIPTION:
SOUTH GRAPE CREEK 69.0
END DESCRIPTION:
XS GIS Cut Line= 4
      2786535.92     10028664.38      2786322.37      10027700.8
      2785884.87     10027023.72      2785916.12      10025789.3
#Sta/Elev= 30
  3390.5 1663.36  3632.4 1653.97  3800.9 1650.17    3817 1646.79  3865.7 1648.68
  3923.8 1647.93  4142.7 1637.37  4186.3 1630.87  4261.8 1627.59  4435.1 1626.22
  4471.4 1622.34  4507.7  1625.3  4522.8 1623.42    4538 1624.76  4543.9 1626.98
  4559.1 1624.61  4565.1 1627.23  4580.2 1628.12  4855.3 1628.26  4891.6 1627.32
  4906.8 1622.18  4912.7 1618.21  4927.9 1613.11  5000.2 1606.45    5079 1618.28
  5115.3 1621.34  5363.6 1621.43  5793.8 1629.85  6073.9  1639.9  6418.4  1649.5
#Mann= 4 ,-1 , 0
  3390.5     .16       0  4912.7     .07       0    5079     .16       0
  6418.4     .05       0
#XS Ineff= 1 ,-1
 4214.32 4608.071628.299
Permanent Ineff=
       T
Bank Sta=4912.7,5079
XS Rating Curve= 0 ,0
Exp/Cntr=0.3,0.1

Type RM Length L Ch R = 1 ,44838   ,560,560,560
BEGIN DESCRIPTION:
SOUTH GRAPE CREEK 68.0
END DESCRIPTION:
XS GIS Cut Line= 3
      2787233.81     10028403.89        2786088.     10026487.26
      2785978.73       10025738.
#Sta/Elev= 30
  3203.9  1643.4  3212.1 1643.53  3296.7 1635.63    3409 1632.35  3771.4  1626.6
  4135.2 1626.19  4242.1 1621.92  4349.2  1621.7  4350.2 1621.66  4374.4  1618.3
  4497.3 1624.58  4699.9 1624.91  4862.7 1622.97  4884.1 1621.68  4905.5 1614.51
  4908.6 1613.67  4928.4 1610.16    4992 1607.06  4994.7 1606.56    4998 1607.06
  5026.1 1608.72  5059.2 1614.08  5245.5 1622.77  5291.4 1625.19  5428.8 1630.99
  5579.7 1631.48  5652.7 1636.26  5713.4 1635.45  5820.5 1639.56  6194.1    1652
#Mann= 17 ,-1 , 0
  3203.9     .05       0  3212.1     .16       0    3409      .1       0
  3771.4     .05       0  4349.2      .1       0  4350.2     .16       0
  4699.9      .1       0  4908.6     .16       0    4992     .07       0
    4998     .16       0  5026.1      .1       0  5245.5     .16       0
  5291.4      .1       0  5428.8     .16       0  5579.7     .05       0
  5713.4      .1       0  5820.5     .05       0
#XS Ineff= 1 ,-1
  4135.4 4541.081625.394
Permanent Ineff=
       T
Bank Sta=4905.5,5059.2
XS Rating Curve= 0 ,0
Exp/Cntr=0.3,0.1

Type RM Length L Ch R = 1 ,44278   ,610,610,610
BEGIN DESCRIPTION:
SOUTH GRAPE CREEK 67.0
END DESCRIPTION:
XS GIS Cut Line= 3
      2787465.73     10027747.24      2787395.29     10027523.72
      2786542.12     10026197.14
#Sta/Elev= 30
    3565 1627.36  3610.8 1623.13  3631.6 1624.54  3652.6 1621.35  3715.5  1619.3
  4182.6 1621.82  4318.4  1623.2  4367.8 1622.08  4728.7 1614.65    4849 1609.41
  4869.2 1607.98  4890.3 1610.08  4940.7 1609.07  4953.7 1607.84  4976.4 1602.72
  4999.9 1601.93  5002.3 1601.69    5005 1601.19  5008.3 1601.69  5041.6 1609.01
  5047.7 1612.04  5071.5    1617    5099 1617.32  5123.9 1622.86  5171.7 1630.89
  5192.8 1640.05    5238 1640.25  5244.3 1643.19  5273.6 1646.16  5376.6 1649.54
#Mann= 9 ,-1 , 0
    3565      .1       0  4182.6     .05       0  4367.8     .16       0
  4728.7     .05       0    4849      .1       0  4999.9     .16       0
  5002.3     .07       0  5008.3     .16       0  5123.9      .1       0
Bank Sta=4940.7,5041.6
XS Rating Curve= 0 ,0
Exp/Cntr=0.3,0.1

Type RM Length L Ch R = 1 ,43668   ,830,830,830
BEGIN DESCRIPTION:
SOUTH GRAPE CREEK 66.0
END DESCRIPTION:
XS GIS Cut Line= 4
      2787503.95     10027754.19      2787577.58     10027539.34
      2787322.37     10026528.92      2787317.17     10025998.22
#Sta/Elev= 30
  3575.3 1627.13  3608.7  1627.2  3660.4 1622.08  3681.5 1623.38  3702.6  1620.7
  3857.3 1618.02  4359.5 1617.94  4437.4 1617.61    4591  1612.2  4705.6 1611.87
  4760.3 1609.91  4796.2 1604.38    4819 1603.67  4879.8 1606.59  4939.8 1606.91
  4969.8 1601.54  5006.5 1600.28  5006.8 1600.27  5009.5 1599.77  5012.8 1600.27
  5039.8 1605.85  5049.8 1610.63  5069.8 1620.08  5109.8 1630.12  5169.8 1639.75
  5203.3 1641.63  5239.8 1640.44  5279.8 1647.71  5299.8 1649.49  5375.3 1649.17
#Mann= 7 ,-1 , 0
  3575.3      .1       0  4359.5     .05       0  4705.6      .1       0
  5006.5     .16       0  5006.8     .07       0  5012.8     .16       0
  5203.3      .1       0
Bank Sta=4939.8,5049.8
XS Rating Curve= 0 ,0
Exp/Cntr=0.3,0.1

Type RM Length L Ch R = 1 ,42838   ,604,604,604
BEGIN DESCRIPTION:
SOUTH GRAPE CREEK 65.0
END DESCRIPTION:
XS GIS Cut Line= 3
      2787817.17      10027643.5      2787957.79     10026940.38
      2787921.33     10026289.34
#Sta/Elev= 30
  4166.6 1618.89  4506.3 1616.67  4579.5 1614.24  4635.5 1613.29  4667.8 1611.32
  4686.5 1609.33  4705.2 1611.23  4756.2 1612.82  4778.2 1611.98  4807.2 1605.86
  4850.9 1608.81  4863.3 1608.37  4879.4 1605.28  4900.3  1603.5  4907.2    1603
  4930.4  1602.2  4958.2  1599.2  4997.5  1598.7  5000.2  1598.2  5003.5  1598.7
  5020.5 1598.91  5070.6 1603.29  5110.6 1606.81  5130.7 1611.47  5150.7 1618.11
  5180.8 1622.49  5270.9 1628.86  5322.3 1635.54  5431.7 1640.84  5535.7 1645.87
#Mann= 8 ,-1 , 0
  4166.6     .05       0  4579.5      .1       0  4667.8     .05       0
  4850.9      .1       0  4907.2     .16       0  4997.5     .07       0
  5003.5     .16       0  5431.7      .1       0
Bank Sta=4900.3,5070.6
XS Rating Curve= 0 ,0
Exp/Cntr=0.3,0.1

Type RM Length L Ch R = 1 ,42234   ,670,670,670
BEGIN DESCRIPTION:
SOUTH GRAPE CREEK 64.0
END DESCRIPTION:
XS GIS Cut Line= 3
      2788499.46     10027883.09      2788473.41     10027127.88
       2788775.5     10025841.43
#Sta/Elev= 30
  4109.1 1627.74  4648.8 1621.89  4728.8  1618.7  4788.7 1611.86  4869.6 1603.83
  4889.6 1605.89  4899.8 1605.06  4906.9    1601  4920.4 1597.48  4949.3 1594.89
  4958.5 1590.21  4961.2 1589.71  4964.5 1590.21  5023.1 1591.89  5053.9 1595.47
  5074.5 1600.27  5089.2 1600.37  5171.6 1602.31  5228.5 1609.05  5279.9 1611.38
  5372.3 1614.08  5427.8 1613.89    5737 1617.27  5803.8 1617.54  5918.4 1622.09
  6045.6  1632.3  6060.6 1632.31  6127.5 1640.53    6178 1643.32  6186.2 1645.25
#Mann= 8 ,-1 , 0
  4109.1     .05       0  4788.7      .1       0  4958.5     .07       0
  4964.5      .1       0  5089.2     .16       0  5427.8      .1       0
    5737     .16       0  6127.5      .1       0
Bank Sta=4906.9,5074.5
XS Rating Curve= 0 ,0
Exp/Cntr=0.3,0.1

Type RM Length L Ch R = 1 ,41564   ,1082,1082,1082
BEGIN DESCRIPTION:
SOUTH GRAPE CREEK 63.0
END DESCRIPTION:
XS GIS Cut Line= 3
      2789056.75     10027867.47      2789192.16     10026841.42
      2789061.96      10025763.3
#Sta/Elev= 30
  4238.3 1620.18  4298.3 1619.34  4474.1 1613.37  4492.8 1614.02  4625.4  1610.4
  4896.9 1609.79  4917.9 1607.18  4940.8 1601.75  4958.2 1596.38  4977.5 1591.62
  4980.2 1591.12  4983.5 1591.62  5018.7 1592.69  5028.8 1595.31  5048.9 1597.03
  5119.6 1597.09    5160 1601.28  5351.5 1607.13  5572.2    1608  5582.8 1607.97
  5898.7 1610.34  5951.4 1611.71  6030.3 1613.16  6147.2 1616.03  6237.9 1623.35
  6263.1 1629.46  6288.3 1633.34  6318.5 1640.81  6345.1 1650.27  6359.2 1652.98
#Mann= 11 ,-1 , 0
  4238.3      .1       0  4298.3     .05       0  4492.8      .1       0
  4940.8     .16       0  4977.5     .07       0  4983.5     .16       0
  5572.2      .1       0  5582.8     .05       0  5898.7      .1       0
  5951.4     .05       0  6030.3     .16       0
Bank Sta=4958.2,5048.9
XS Rating Curve= 0 ,0
Exp/Cntr=0.3,0.1

Type RM Length L Ch R = 1 ,40482   ,332,332,332
BEGIN DESCRIPTION:
SOUTH GRAPE CREEK 62.0
END DESCRIPTION:
XS GIS Cut Line= 3
      2789697.37     10028206.01      2790186.96     10027393.51
      2790358.84      10026471.6
#Sta/Elev= 30
  3961.6 1617.13  4000.8 1614.89  4180.3 1604.07  4247.5 1601.91  4491.6 1602.05
  4606.4 1601.78  4734.9 1597.95  4793.2 1600.36  4818.1 1596.52  4927.8 1592.95
  4940.5 1592.42    4971 1589.23  4991.4 1582.39  5000.5 1581.68  5003.2 1581.18
  5006.5 1581.68    5032 1588.02  5072.7 1593.14  5097.3 1594.73  5166.7 1594.13
  5184.6 1597.81  5214.3 1608.61  5219.4 1608.07  5255.8 1621.65  5272.1 1625.63
  5337.2 1634.18  5382.6 1637.36  5398.3 1641.42  5451.6 1643.36    5848 1651.47
#Mann= 10 ,-1 , 0
  3961.6      .1       0  4000.8     .05       0  4180.3      .1       0
  4491.6     .05       0  4818.1      .1       0  4927.8     .05       0
  5000.5    .035       0  5006.5     .05       0  5097.3     .16       0
  5451.6      .1       0
Bank Sta=4940.5,5072.7
XS Rating Curve= 0 ,0
Exp/Cntr=0.3,0.1

Type RM Length L Ch R = 1 ,40150   ,556,556,556
BEGIN DESCRIPTION:
SOUTH GRAPE CREEK 61.0
END DESCRIPTION:
XS GIS Cut Line= 3
      2789926.55     10028221.62      2790582.79     10027299.76
      2790587.99     10026597.66
#Sta/Elev= 30
    4090 1615.92  4154.3 1611.84  4204.7 1606.26    4247 1604.62  4283.8 1605.03
  4305.5 1601.24  4343.1 1599.62  4524.2 1595.82  4786.3 1596.56    4849 1591.37
    4876 1590.93    4908 1592.49  4943.7 1590.09  4964.6 1584.57  4993.2 1583.32
    5012 1582.27  5014.7 1581.77    5018 1582.27  5029.8 1584.04  5035.9 1589.38
  5044.5 1594.29  5050.7 1598.65  5057.1  1600.6  5067.6 1600.81  5174.3 1599.36
  5337.6 1601.27  5521.6 1608.77  5593.5 1611.99  5897.6 1630.62  5923.7 1633.81
#Mann= 11 ,-1 , 0
    4090     .05       0  4343.1      .1       0  4524.2     .05       0
    4876      .1       0  4993.2     .16       0    5012     .07       0
    5018     .16       0  5067.6      .1       0  5174.3     .05       0
  5521.6     .16       0  5593.5      .1       0
Bank Sta=4908,5044.5
XS Rating Curve= 0 ,0
Exp/Cntr=0.3,0.1

Type RM Length L Ch R = 1 ,39594   ,506,506,506
BEGIN DESCRIPTION:
SOUTH GRAPE CREEK 60.0
END DESCRIPTION:
XS GIS Cut Line= 3
      2790020.27     10028544.56      2790770.29     10027846.63
      2791207.79     10027028.93
#Sta/Elev= 30
  4195.3  1620.5  4449.5 1611.25  4525.3 1610.56  4659.5 1607.93    4683 1604.38
  4725.5 1591.91  4779.7 1593.66  4845.7 1589.82  4944.4 1589.79  4965.9  1586.9
  4986.9  1579.2    4998 1578.75  4998.1 1578.74  5000.8 1578.24  5004.1 1578.74
  5036.7 1587.02  5057.7 1588.48  5093.4 1595.38  5238.4 1594.23    5663 1594.11
  5687.7 1594.37  5709.6 1590.35  5806.5 1594.15  5923.3 1601.53  5945.3    1605
  5974.5 1614.03    6033 1626.88  6093.2 1636.18  6098.9 1639.24  6147.2 1643.83
#Mann= 11 ,-1 , 0
  4195.3      .1       0  4525.3     .05       0  4659.5     .16       0
  4779.7     .05       0    4998     .16       0  4998.1     .07       0
  5004.1     .16       0  5238.4     .05       0    5663      .1       0
  5806.5     .05       0  5974.5     .16       0
Bank Sta=4965.9,5036.7
XS Rating Curve= 0 ,0
Exp/Cntr=0.3,0.1

Type RM Length L Ch R = 1 ,39088   ,1208,1208,1208
BEGIN DESCRIPTION:
SOUTH GRAPE CREEK 59.0
END DESCRIPTION:
XS GIS Cut Line= 3
      2790874.46     10028898.71      2790973.41     10028133.09
      2791327.57     10027153.96
#Sta/Elev= 30
  4420.8 1608.54  4491.2 1603.82  4631.1 1602.68  4714.8 1602.52  4869.5 1601.44
  4950.1 1596.09  4962.2 1594.36  4970.3 1589.46  4980.4 1582.51  4997.6 1577.49
  5000.3 1576.99  5003.6 1577.49  5030.8 1580.89  5061.1 1579.07  5121.6 1587.99
  5182.1 1592.02  5537.9  1587.4  5664.3 1583.63    5695  1584.1  5720.3 1588.21
  5725.6 1586.38  5794.1  1589.4  5868.3 1590.41  5929.6 1584.42  5954.9 1588.14
  6018.6 1611.59  6077.5 1636.29  6108.2 1642.54  6164.1 1650.47    6234 1652.31
#Mann= 8 ,-1 , 0
  4420.8     .05       0  4631.1      .1       0  4714.8     .05       0
  4997.6     .04       0  5003.6     .05       0  5537.9      .1       0
  5794.1     .05       0  6018.6     .16       0
Bank Sta=4970.3,5121.6
XS Rating Curve= 0 ,0
Exp/Cntr=0.3,0.1

Type RM Length L Ch R = 1 ,37880   ,571,571,571
BEGIN DESCRIPTION:
SOUTH GRAPE CREEK 58.0
END DESCRIPTION:
XS GIS Cut Line= 3
      2791280.71     10029008.07      2791431.75     10027810.17
      2791706.88     10027467.55
#Sta/Elev= 30
  3690.6 1602.81  3836.1 1598.41    3877 1592.54  3946.7 1592.03  4397.4 1590.99
  4561.8 1589.66  4692.8 1585.52  4733.1 1585.68  4799.5 1588.17  4900.3 1586.62
  4929.1 1582.11  4935.5 1579.12  4949.9 1576.31  5003.6 1575.51  5018.7 1575.35
  5021.4 1574.85  5024.7 1575.35  5049.1 1579.56  5057.1 1582.23  5063.5  1586.8
  5077.9 1594.04  5092.3 1597.68  5141.9 1625.48  5156.3 1631.77  5170.7 1642.25
  5185.1 1645.14  5234.7 1650.38  5277.9 1653.37  5302.5 1653.76  5337.4 1654.44
#Mann= 8 ,-1 , 0
  3690.6     .05       0  3946.7      .1       0  4397.4     .05       0
  4799.5      .1       0  5003.6     .16       0  5018.7     .07       0
  5024.7     .16       0  5302.5      .1       0
Bank Sta=4929.1,5057.1
XS Rating Curve= 0 ,0
Exp/Cntr=0.3,0.1

Type RM Length L Ch R = 1 ,37309   ,432,432,432
BEGIN DESCRIPTION:
SOUTH GRAPE CREEK 57.0
END DESCRIPTION:
XS GIS Cut Line= 3
      2791457.77     10029086.26      2791817.16      10028263.3
      2791890.07     10027732.09
#Sta/Elev= 30
  3915.2 1598.07  3994.3  1592.1  4048.9 1590.89  4124.6 1591.56  4182.3 1590.68
  4229.1 1591.04  4853.1 1586.68  4893.5 1579.33  4913.7 1577.32  4954.1 1573.93
  4974.3 1573.04  5007.9 1568.78  5014.6 1569.99  5034.8 1569.71  5044.9 1570.66
  5095.4 1577.52  5125.7 1578.75  5157.4 1581.38  5176.1 1584.69  5206.4 1597.51
  5224.4  1603.9  5229.5 1602.65  5236.7 1605.23  5287.2 1618.35  5296.5 1622.77
  5301.6 1620.98  5307.4 1624.19  5317.5 1627.42  5346.1 1635.18  5349.4 1635.18
#Mann= 4 ,-1 , 0
  3915.2      .1       0  4913.7     .07       0  5095.4      .1       0
  5349.4     .16       0
Bank Sta=4913.7,5095.4
XS Rating Curve= 0 ,0
Exp/Cntr=0.3,0.1

Type RM Length L Ch R = 1 ,36877   ,470,470,470
BEGIN DESCRIPTION:
SOUTH GRAPE CREEK 56.0
END DESCRIPTION:
XS GIS Cut Line= 3
      2791608.81     10029325.83      2792233.83     10028320.59
      2792353.47     10027628.76
#Sta/Elev= 30
  3673.6 1595.96  3782.5 1589.58  4117.8 1588.95    4459 1584.08  4669.2 1584.27
  4884.6 1573.56  4911.9 1575.63  4985.8 1563.89  5026.4 1567.47  5036.8 1570.42
  5046.9 1583.14  5057.1  1588.6    5118 1589.53  5178.9 1583.01  5210.8 1586.42
  5239.8 1585.09  5280.4 1587.06  5325.3 1591.28  5351.4 1596.51  5361.5 1600.71
  5371.7 1609.38    5380 1612.44  5385.1 1612.32  5402.1 1603.84  5444.9 1602.63
  5452.9 1605.75  5473.2 1621.58  5483.3 1626.24  5513.8 1633.08  5559.4 1646.76
#Mann= 4 ,-1 , 0
  3673.6      .1       0  4911.9     .07       0  5036.8      .1       0
  5559.4     .16       0
Bank Sta=4911.9,5036.8
XS Rating Curve= 0 ,0
Exp/Cntr=0.3,0.1

Type RM Length L Ch R = 1 ,36407   ,801,801,801
BEGIN DESCRIPTION:
Mapping XS bf49d6e4
END DESCRIPTION:
XS GIS Cut Line= 4
       2791650.5     10029482.05      2792220.13     10028632.73
      2792806.07     10028502.52      2793261.77     10027864.54
#Sta/Elev= 30
  3804.9 1592.82  4010.6 1588.96  4465.1 1587.98  4550.9 1584.31  4645.7 1583.93
  4673.9 1581.54  4827.6 1579.41  4892.3 1576.96  4940.9 1572.68  4984.5  1567.8
    5010 1562.85  5020.5 1566.51    5028 1572.28  5028.4 1572.23  5033.1 1571.65
    5041 1580.54  5051.2 1585.31  5061.5 1586.41  5212.4 1583.76  5463.5 1587.23
    5493 1588.67  5507.8 1590.94  5536.9 1588.56  5593.8 1591.48  5837.1 1595.86
  6065.7 1603.09  6095.2 1607.51  6130.8 1622.27  6188.2 1637.21  6211.8 1639.49
#Mann= 4 ,-1 , 0
  3804.9      .1       0  4940.9     .07       0  5028.4      .1       0
  6211.8      .1       0
Bank Sta=4940.9,5028
XS Rating Curve= 0 ,0
Exp/Cntr=0.3,0.1

Type RM Length L Ch R = 1 ,35606   ,456,456,456
BEGIN DESCRIPTION:
SOUTH GRAPE CREEK 55.0
END DESCRIPTION:
XS GIS Cut Line= 2
      2791843.17     10029825.82      2794030.06     10028359.27
#Sta/Elev= 30
  4125.9 1599.31  4324.9 1587.89  4765.7 1584.43  4837.7  1577.8  4843.8 1571.59
  4858.8 1570.16  4902.9 1571.44  4930.8 1581.36  4951.8 1582.57  4966.8  1582.7
  4981.8 1575.22  4996.8 1564.23  5002.8 1562.95  5038.8 1564.31  5074.6 1561.25
  5104.8 1563.58  5131.9 1572.29  5312.2 1581.51    5342 1585.92  5384.5 1597.38
    5465 1605.55  5630.1 1610.26  5774.1  1610.4  5903.2 1616.56  6026.2 1613.19
  6149.3 1598.44  6323.3 1598.17  6545.4 1610.25  6689.5  1623.5    6759 1636.39
#Mann= 4 ,-1 , 0
  4125.9      .1       0  4981.8     .07       0  5131.9      .1       0
    6759     .16       0
Bank Sta=4981.8,5131.9
XS Rating Curve= 0 ,0
Exp/Cntr=0.3,0.1

Type RM Length L Ch R = 1 ,35150   ,308,308,308
BEGIN DESCRIPTION:
SOUTH GRAPE CREEK 54.0
END DESCRIPTION:
XS GIS Cut Line= 3
      2792192.17     10030112.25      2792843.21     10029690.38
      2794015.88     10028607.73
#Sta/Elev= 30
    4104  1591.7  4266.4 1591.21  4635.8  1582.4  4923.7  1581.4  4944.7 1578.43
  4958.8 1574.17  4966.2 1569.16  4980.4 1560.91  4994.3 1557.17  5043.9 1566.98
  5079.1 1568.99  5114.8 1568.32  5298.5 1581.89  5525.3 1585.55  5560.5 1589.46
  5645.5    1589  5666.5 1593.51  5673.9  1592.3  5680.7  1595.7  5688.1 1594.66
  5694.9 1598.12  5716.4 1597.59  5723.2 1600.45  5737.4  1600.9  5956.8 1591.05
  6190.5 1595.14  6303.3 1603.26  6388.4 1613.52  6409.9 1619.32  6475.8 1626.02
#Mann= 4 ,-1 , 0
    4104     .16       0  4966.2     .07       0  5079.1     .16       0
  6475.8      .1       0
Bank Sta=4966.2,5079.1
XS Rating Curve= 0 ,0
Exp/Cntr=0.3,0.1

Type RM Length L Ch R = 1 ,34842   ,751,751,751
BEGIN DESCRIPTION:
SOUTH GRAPE CREEK 53.0
END DESCRIPTION:
XS GIS Cut Line= 2
      2792666.15     10030310.14      2794199.33     10028762.91
#Sta/Elev= 30
  4275.4 1585.77  4451.3 1584.79  4656.3 1580.13  4889.7 1578.03  4917.9 1576.22
  4953.3 1568.17  4967.5 1566.03  4981.6 1561.26  5009.6 1557.44  5012.9 1557.94
    5024 1565.61  5052.3 1567.94  5059.4 1566.37  5066.5 1568.04  5144.2    1570
  5179.6 1573.37  5214.9 1579.39  5243.2 1580.33  5865.5 1585.38  5922.1 1586.19
  6056.4 1591.72  6120.1 1592.23  6148.3 1595.27    6212 1608.62  6268.6 1612.34
  6303.2 1612.94  6346.3 1621.08  6388.8 1622.82  6445.3 1627.32  6453.6 1629.23
#Mann= 4 ,-1 , 0
  4275.4     .16       0  4953.3     .07       0  5052.3     .16       0
  6453.6      .1       0
Bank Sta=4953.3,5052.3
XS Rating Curve= 0 ,0
Exp/Cntr=0.3,0.1

Type RM Length L Ch R = 1 ,34091   ,836,836,836
BEGIN DESCRIPTION:
SOUTH GRAPE CREEK 52.0
END DESCRIPTION:
XS GIS Cut Line= 3
      2793395.29     10031804.97      2793681.75     10030315.38
      2794472.73     10029227.78
#Sta/Elev= 30
  3352.1 1595.01  3449.2 1593.23  3577.4 1584.69    3669 1582.01  3921.7 1581.11
  4300.6 1582.24  4707.7 1577.11  4758.7  1571.6  4830.1 1567.24  4918.6 1564.18
  4945.7 1558.49  4968.8 1559.78  5004.1 1554.77  5019.1 1558.75  5031.8 1567.01
  5046.1  1571.3  5075.5 1574.69  5211.5 1574.52    5312 1577.25    5448 1577.26
  5498.2 1578.97  5575.8 1577.87  5820.5 1581.04  5897.8 1580.33  6048.5 1583.84
  6092.5 1586.96  6148.9 1594.15  6178.3 1596.23  6199.2  1605.7  6213.8 1609.57
#Mann= 4 ,-1 , 0
  3352.1     .16       0  4918.6     .07       0  5031.8     .16       0
  6213.8     .16       0
Bank Sta=4918.6,5031.8
XS Rating Curve= 0 ,0
Exp/Cntr=0.3,0.1

Type RM Length L Ch R = 1 ,33255   ,879,879,879
BEGIN DESCRIPTION:
SOUTH GRAPE CREEK 51.0
END DESCRIPTION:
XS GIS Cut Line= 4
      2793624.43     10031914.38      2794504.66     10030336.22
      2794280.71     10029601.84      2794562.77     10029297.99
#Sta/Elev= 30
  2947.9 1595.06  3040.2 1592.27  3155.8 1582.75  3258.7  1580.3  3361.5 1579.16
  3692.9 1580.83  4178.6 1577.61  4508.9 1571.46  4897.4 1575.94  4924.8  1571.3
  4930.3 1567.99  4977.1 1555.25  4995.6 1553.76  5018.9 1554.87  5050.3 1561.17
  5123.5 1568.12  5154.8 1572.89  5203.3 1575.99  5301.2 1574.38  5569.4 1578.31
  5604.5 1575.13  5640.2 1579.39  5717.9 1580.32  5781.4 1583.36  5817.1  1588.6
  5838.1 1595.18  5859.6 1596.92  5873.8 1600.46  5902.1 1610.72  5937.3 1626.65
#Mann= 4 ,-1 , 0
  2947.9     .16       0  4930.3     .07       0  5123.5     .16       0
  5937.3     .16       0
#XS Ineff= 1 ,-1
 4237.21 4896.97 1576.23
Permanent Ineff=
       T
Bank Sta=4930.3,5123.5
XS Rating Curve= 0 ,0
Exp/Cntr=0.3,0.1

Type RM Length L Ch R = 1 ,32376   ,684,684,684
BEGIN DESCRIPTION:
SOUTH GRAPE CREEK 50.0
END DESCRIPTION:
XS GIS Cut Line= 2
      2793702.59     10031935.16      2795462.99     10029794.56
#Sta/Elev= 30
  2559.7 1593.91  2621.9 1590.94  2728.8 1582.04  2848.7 1578.81  3076.8 1579.99
  3850.9 1575.75  4198.9 1568.57  4462.2 1572.66  4767.1 1569.83  4866.2 1565.62
  4958.7 1558.06  5001.5 1549.21  5030.4 1550.95  5065.6 1558.98  5079.9 1559.77
  5094.3 1564.23  5108.6 1575.18    5123 1583.15  5158.1 1596.65  5207.6 1609.53
  5215.5 1613.99    5222 1614.75  5236.3  1623.7  5242.8  1623.3  5250.7 1627.29
  5257.1 1627.13    5265 1632.12  5271.5 1632.15  5279.4 1635.62  5331.2 1639.92
#Mann= 3 ,-1 , 0
  2559.7     .16       0  4866.2     .07       0  5094.3     .16       0
#XS Ineff= 1 ,-1
 3967.19 4459.38 1572.79
Permanent Ineff=
       T
Bank Sta=4866.2,5094.3
XS Rating Curve= 0 ,0
Exp/Cntr=0.3,0.1

Type RM Length L Ch R = 1 ,31692   ,466,466,466
BEGIN DESCRIPTION:
SOUTH GRAPE CREEK 49.0
END DESCRIPTION:
XS GIS Cut Line= 3
      2793723.39      10031940.4      2795207.79     10030653.92
       2795869.3     10030653.92
#Sta/Elev= 30
  2858.2 1592.81  2930.8 1589.41  3015.3 1582.04  3121.6 1578.84  3248.9 1579.84
  3915.6 1576.82  4036.2 1575.23  4156.9 1570.73  4496.8 1566.11    4759 1570.06
  4809.3 1566.37  4903.2  1564.8  4933.2 1560.06  4963.2 1551.49  4973.2 1547.16
  4982.9 1546.07  5033.2 1550.54  5053.2 1555.42  5063.2 1560.21  5083.2 1575.24
  5103.2 1587.09  5113.2 1591.74  5133.2 1596.03  5143.2 1600.73  5193.2 1628.25
  5213.2 1644.33  5223.2 1648.43  5333.2  1656.7  5383.2 1665.81    5484 1675.47
#Mann= 4 ,-1 , 0
  2858.2     .16       0  4933.2     .07       0  5063.2     .16       0
    5484      .1       0
Bank Sta=4933.2,5063.2
XS Rating Curve= 0 ,0
Exp/Cntr=0.3,0.1

Type RM Length L Ch R = 1 ,31226   ,644,644,644
BEGIN DESCRIPTION:
SOUTH GRAPE CREEK 48.0
END DESCRIPTION:
XS GIS Cut Line= 3
      2793791.13     10031950.79      2795186.96     10031112.26
      2795904.54     10030951.06
#Sta/Elev= 30
  3296.5 1589.41  3496.1 1578.33  4269.5 1577.64    4423 1571.39  4809.6  1565.9
  4889.3 1557.28  4910.7 1550.84  4916.5 1553.66  4936.2 1549.94  4941.3 1552.09
  4957.1 1546.74  5008.1 1544.45    5028 1550.33  5081.5 1557.74  5100.6 1561.47
  5119.7 1570.82  5124.8 1570.87  5131.4 1577.02  5168.1 1597.86  5173.3 1596.54
  5211.5 1618.27  5216.6 1617.31  5223.6 1622.82  5259.9 1638.51  5295.4 1641.02
  5315.9 1653.07  5346.5 1659.15  5377.3 1669.17  5438.3 1676.19  5660.3 1678.42
#Mann= 4 ,-1 , 0
  3296.5     .16       0  4889.3     .07       0  5081.5     .16       0
  5660.3     .16       0
Bank Sta=4889.3,5081.5
XS Rating Curve= 0 ,0
Exp/Cntr=0.3,0.1

Type RM Length L Ch R = 1 ,30582   ,470,470,470
BEGIN DESCRIPTION:
SOUTH GRAPE CREEK 47.0
END DESCRIPTION:
XS GIS Cut Line= 3
      2793853.65     10032002.88      2795442.16     10031653.92
      2796034.73     10031310.86
#Sta/Elev= 30
  3601.3 1582.34  3713.8 1577.97  3762.7 1577.37  3806.5 1574.87  4035.6    1574
  4374.1 1576.17  4547.9 1571.89  4650.8 1572.42  4787.3 1570.31    4880 1566.06
  4928.9 1561.62  4957.7 1554.69  4967.5 1551.28  4972.7  1551.4  4988.4  1545.1
  5008.7 1544.32  5039.6 1546.18  5049.9  1549.4  5070.5 1551.22  5090.8 1554.81
  5131.8 1555.58  5201.8 1560.29  5260.9 1562.62  5276.7  1564.7  5431.4 1567.15
    5651 1575.71  5766.5 1585.08  5833.4  1593.4  5860.8 1598.06  5912.4 1602.89
#Mann= 4 ,-1 , 0
  3601.3     .16       0  4957.7     .07       0  5090.8     .16       0
  5912.4     .16       0
Bank Sta=4957.7,5090.8
XS Rating Curve= 0 ,0
Exp/Cntr=0.3,0.1

Type RM Length L Ch R = 1 ,30112   ,441,441,441
BEGIN DESCRIPTION:
SOUTH GRAPE CREEK 46.0
END DESCRIPTION:
XS GIS Cut Line= 4
     2794051.822    10032033.133     2795062.238    10031814.383
     2795149.053    10032156.694     2796791.122    10031867.466
#Sta/Elev= 30
       01576.053249.1567 1573.16368.75191574.726 558.1111575.088727.53751571.291
847.13271570.495877.03151568.634976.6942 1568.551134.7441564.1321400.1421562.989
1439.9181560.2441459.8051556.3511469.7491551.9581479.6931547.4871489.6371544.634
 1499.581543.6181618.9061550.9581678.5691551.7181698.4571553.7671728.2881559.237
1827.7261562.3552364.6911563.6452563.5681567.3892672.9491572.0292732.6121576.901
2861.8821592.4472901.6571601.593 2961.321622.8063020.9831634.0933050.8141636.793
#Mann= 3 ,-1 , 0
       0     .16       01469.749     .07       01618.906     .16       0
Bank Sta=1469.749,1618.906
XS Rating Curve= 0 ,0
Exp/Cntr=0.3,0.1

Type RM Length L Ch R = 1 ,29671   ,375,375,375
BEGIN DESCRIPTION:
SOUTH GRAPE CREEK 45.0
END DESCRIPTION:
XS GIS Cut Line= 3
       2794530.7     10033169.56      2794916.12     10032690.38
      2796701.85     10032138.53
#Sta/Elev= 30
  3987.2  1576.5  4217.1 1566.69  4373.9 1562.92  4409.1  1564.1  4537.1 1556.31
  4646.7 1553.15  4730.2 1546.54  4815.1 1556.17    4913 1556.29  4950.8 1552.41
  4970.9 1542.08  5015.8 1540.58  5043.5 1546.93  5086.6 1549.15    5107 1547.62
  5146.6 1552.12  5151.9 1551.66  5179.3 1557.82  5211.7 1560.58  5441.9 1564.49
  5760.2 1558.98  5954.8 1559.34  6153.7 1563.98    6206 1567.43  6226.9  1567.1
  6247.9 1570.42  6330.7 1577.28  6368.6 1584.62  6425.8 1589.41  6471.2 1596.65
#Mann= 4 ,-1 , 0
  3987.2     .16       0  4950.8     .07       0  5146.6     .16       0
  6471.2      .1       0
#XS Ineff= 2 ,-1
  4435.8 4863.64  1556.9 5445.31 6185.94 1564.62
Permanent Ineff=
       T       T
Bank Sta=4950.8,5146.6
XS Rating Curve= 0 ,0
Exp/Cntr=0.3,0.1

Type RM Length L Ch R = 1 ,29296   ,220,220,220
BEGIN DESCRIPTION:
SOUTH GRAPE CREEK 43.0
END DESCRIPTION:
XS GIS Cut Line= 3
      2794546.37     10033221.62      2796291.12     10032518.51
      2796900.52     10032112.24
#Sta/Elev= 30
  4250.4 1578.06  4360.1 1576.36  4521.2 1568.25    4533 1565.65  4597.7 1560.74
  4640.8 1553.52  4682.4 1553.48  4813.3 1543.34  4819.3 1546.28  4843.5 1548.01
  4910.3 1548.41  4926.7 1543.94  4932.1 1546.27  4950.9 1543.14  5033.9 1540.57
  5037.2 1541.07  5039.7 1544.05  5058.3 1548.41  5087.9 1548.47    5112 1553.73
  5117.4 1552.26  5136.2 1557.04  5189.9 1562.44  5804.8 1560.06  5917.6 1562.06
  6140.3 1558.23    6298 1561.61  6523.3 1574.28  6817.8 1608.17  6863.9 1611.81
#Mann= 4 ,-1 , 0
  4250.4     .16       0  4910.3     .07       0  5058.3     .16       0
  6863.9      .1       0
#XS Ineff= 2 ,-1
  4714.2 4845.45 1548.11 5919.53 6390.62 1562.23
Permanent Ineff=
       T       T
Bank Sta=4910.3,5058.3
XS Rating Curve= 0 ,0
Exp/Cntr=0.3,0.1

Type RM Length L Ch R = 1 ,29076   ,458,458,458
BEGIN DESCRIPTION:
Mapping XS 78a7bacf
END DESCRIPTION:
XS GIS Cut Line= 3
      2794572.35      10033383.1      2796390.08     10032659.13
      2796910.93     10032263.29
#Sta/Elev= 30
  4355.3 1580.84  4577.2  1577.4  4612.6 1570.54    4631 1570.71  4636.9 1574.39
  4652.5 1574.96  4666.5 1572.25  4684.8 1564.48  4690.8 1560.05  4727.9  1551.8
  4750.1 1549.37  4889.3 1543.16  4965.6 1542.07  5050.8 1542.69  5092.6 1549.24
    5098 1548.15  5127.7 1557.38  5169.2 1560.94  5750.6 1560.12  6230.7 1556.04
  6328.9 1557.52  6399.6 1561.61  6507.7 1560.84    6593 1563.56  6628.4 1567.12
  6757.3 1573.06  6792.6 1577.12  6871.6  1581.3  6892.5    1586  6966.1 1592.88
#Mann= 4 ,-1 , 0
  4355.3     .16       0  4750.1     .07       0  5092.6     .16       0
  6966.1      .1       0
#XS Ineff= 1 ,-1
 5382.81 6763.28 1561.13
Permanent Ineff=
       T
Bank Sta=4750.1,5092.6
XS Rating Curve= 0 ,0
Exp/Cntr=0.3,0.1

Type RM Length L Ch R = 1 ,28618   ,587,587,587
BEGIN DESCRIPTION:
SOUTH GRAPE CREEK 44.0
END DESCRIPTION:
XS GIS Cut Line= 3
      2794535.88     10033768.52      2795530.71     10033461.22
      2796968.21     10032523.71
#Sta/Elev= 30
  4370.8 1584.69  4635.2 1582.29  4729.4  1577.1  4771.2 1572.67  4792.2  1568.7
  4802.6 1566.01  4809.2 1562.05  4814.4 1561.23    4834  1552.5    4855 1547.79
  4907.1 1542.63    4945 1541.27  4970.1 1542.71  5001.2 1538.97  5074.7 1541.45
  5118.7 1546.29  5146.1 1551.82  5189.9 1556.86  5458.1  1558.9  5711.6 1559.09
  5922.7 1556.75  6441.9 1555.62  6507.7 1557.02  6550.5 1554.48  6710.5 1554.14
  6933.7 1559.17  7027.3 1562.89  7048.3 1566.01  7099.7 1566.06  7128.2 1568.75
#Mann= 4 ,-1 , 0
  4370.8     .16       0    4855     .07       0  5118.7     .16       0
  7128.2     .05       0
#XS Ineff= 1 ,-1
 5659.77 7059.77 1559.27
Permanent Ineff=
       T
Bank Sta=4855,5118.7
XS Rating Curve= 0 ,0
Exp/Cntr=0.3,0.1

Type RM Length L Ch R = 1 ,28031   ,459,459,459
BEGIN DESCRIPTION:
Mapping XS eaff9f1a
END DESCRIPTION:
XS GIS Cut Line= 2
      2794791.09     10034325.82      2797140.07     10032659.14
#Sta/Elev= 30
  4391.9 1583.82  4699.6 1581.49  4750.1 1578.48  4800.5 1578.25    4851 1574.97
  4857.1 1572.59  4865.7 1573.25  4886.7 1570.03  4907.6 1560.68  4937.1 1552.11
    4958 1543.61  4972.8 1536.59  4978.9 1530.98  4987.5 1527.99  5001.5 1526.64
  5050.8 1534.28  5087.6 1536.02  5136.6 1542.33  5165.9 1544.03  5259.3  1555.5
  5933.6 1557.71  6285.4 1554.92  6436.4 1555.57  6457.7 1553.46    6529 1552.58
  6837.8 1552.55  7096.2  1557.1    7218 1562.58  7245.6 1566.43  7272.1 1566.12
#Mann= 4 ,-1 , 0
  4391.9     .16       0    4958     .07       0  5136.6     .16       0
  7272.1     .05       0
#XS Ineff= 1 ,-1
 5941.41 7281.25 1557.66
Permanent Ineff=
       T
Bank Sta=4958,5136.6
XS Rating Curve= 0 ,0
Exp/Cntr=0.3,0.1

Type RM Length L Ch R = 1 ,27572   ,742,742,742
BEGIN DESCRIPTION:
SOUTH GRAPE CREEK 42.0
END DESCRIPTION:
XS GIS Cut Line= 2
      2795233.86      10034591.4      2797404.59     10032852.73
#Sta/Elev= 30
    4522 1578.72  4643.9 1577.81  4672.7 1575.19  4786.4 1570.06  4872.8 1571.79
  4879.2 1569.76  4893.6 1569.31    4900 1565.34    4908    1563  4914.4 1557.62
  4922.4 1554.64  4943.2 1541.99    4964 1533.85    4972 1533.04  4986.4 1526.87
  5000.6 1525.93  5036.1 1532.69  5100.1 1537.28  5120.9 1541.27  5135.3 1544.63
  5156.1 1546.86  5242.5 1550.77    6046 1555.81  6138.9 1554.02  6593.4 1552.55
  6828.7 1549.11    7064 1552.54  7091.2 1554.27  7163.2 1564.31  7303.2 1566.51
#Mann= 4 ,-1 , 0
    4522     .16       0  4943.2     .07       0  5120.9     .16       0
  7303.2      .1       0
#XS Ineff= 1 ,-1
 6042.19 7178.91 1555.96
Permanent Ineff=
       T
Bank Sta=4943.2,5120.9
XS Rating Curve= 0 ,0
Exp/Cntr=0.3,0.1

Type RM Length L Ch R = 1 ,26830   ,406,406,406
BEGIN DESCRIPTION:
SOUTH GRAPE CREEK 41.0
END DESCRIPTION:
XS GIS Cut Line= 4
      2795973.43     10034700.78      2796218.21      10034388.3
      2796499.46     10033747.67      2797520.31     10032830.99
#Sta/Elev= 30
  4437.5 1568.68  4738.6 1562.46  4759.8 1559.57  4846.2 1559.35  4898.4 1552.69
  4915.9 1544.25  4921.7 1538.77  4927.2 1540.41  4937.7 1535.41  4945.1 1530.77
  4950.6 1531.96  4968.2 1526.41    5036 1527.54    5044 1530.88  5142.9 1535.61
  5223.9 1531.34  5241.8 1534.47  5270.6 1534.85    5294 1546.72  5299.4 1544.69
  5317.3  1549.4  5322.8  1547.5  5340.7 1551.97  5346.2 1550.14    5375  1554.3
    6060 1552.16  6350.8  1548.3  6563.1 1551.88  6661.7 1561.36  6906.1 1568.07
#Mann= 4 ,-1 , 0
  4437.5     .16       0  4937.7     .07       0  5142.9     .16       0
  6906.1     .05       0
#XS Ineff= 1 ,-1
 5396.88 6690.62 1554.17
Permanent Ineff=
       T
Bank Sta=4937.7,5142.9
XS Rating Curve= 0 ,0
Exp/Cntr=0.3,0.1

Type RM Length L Ch R = 1 ,26424   ,535,535,535
BEGIN DESCRIPTION:
SOUTH GRAPE CREEK 40.0
END DESCRIPTION:
XS GIS Cut Line= 3
      2796640.08     10034575.78      2796718.21     10033924.76
      2797603.51     10032914.46
#Sta/Elev= 30
  4619.6 1560.55  4722.4 1558.53  4782.8 1555.19    4803 1551.52  4823.1 1542.37
  4843.2 1542.55  4873.5 1536.77  4904.3 1533.93  4981.5 1524.74  5004.1  1523.8
  5014.5    1525  5034.6  1531.8  5044.7 1532.75  5063.7 1530.63    5085 1526.58
  5105.1  1527.2  5125.3 1531.27    5156 1542.09  5165.5 1543.24  5185.7 1549.05
  5195.8 1550.51  5502.7 1553.18  5665.8  1550.9  5949.5  1550.9  6154.5 1547.24
  6346.2 1552.75  6403.1 1556.25  6452.5 1557.76  6530.3 1563.63  6618.6 1568.17
#Mann= 4 ,-1 , 0
  4619.6     .16       0  4904.3     .07       0  5044.7     .16       0
  6618.6     .05       0
#XS Ineff= 1 ,-1
 5496.09 6445.31  1553.2
Permanent Ineff=
       T
Bank Sta=4904.3,5044.7
XS Rating Curve= 0 ,0
Exp/Cntr=0.3,0.1

Type RM Length L Ch R = 1 ,25889   ,573,573,573
BEGIN DESCRIPTION:
SOUTH GRAPE CREEK 39.0
END DESCRIPTION:
XS GIS Cut Line= 2
      2796947.37     10034862.26      2797723.43     10033049.71
#Sta/Elev= 30
  4356.7 1558.88  4524.2 1559.15  4594.4 1557.33  4735.8 1546.64  4758.2 1546.59
  4805.3 1541.28  4822.9 1536.99  4828.9 1534.34  4866.4 1529.44    4899 1529.89
  4942.5 1524.95  4964.3 1524.11  4986.5 1519.09  5018.7 1521.51  5033.9 1525.16
  5040.4 1530.05  5057.4 1539.93  5062.9 1539.68    5081 1543.38  5086.5 1542.42
    5110 1544.03  5127.4  1547.2  5399.4 1548.56  5714.1 1547.22  5848.3 1545.08
  6076.8 1552.56  6129.4 1552.86  6147.6 1553.99  6182.6 1559.21  6328.4 1564.29
#Mann= 4 ,-1 , 0
  4356.7     .16       0    4899     .07       0  5040.4     .16       0
  6328.4      .1       0
#XS Ineff= 1 ,-1
 5355.77 6054.07 1548.56
Permanent Ineff=
       T
Bank Sta=4899,5040.4
XS Rating Curve= 0 ,0
Exp/Cntr=0.3,0.1

Type RM Length L Ch R = 1 ,25316   ,515,515,515
BEGIN DESCRIPTION:
SOUTH GRAPE CREEK 38.0
END DESCRIPTION:
XS GIS Cut Line= 2
      2797499.44     10035164.38      2798025.51     10033570.56
#Sta/Elev= 30
  4188.3 1553.49  4220.6 1552.87  4273.2 1548.65    4368 1547.23    4726 1546.83
  4768.2 1544.99  4799.8 1541.36  4831.4 1536.84  4869.7 1529.43  4906.7 1525.78
  4957.7 1522.14  4964.9 1520.62  4996.4 1519.19  5010.4 1520.33  5028.4 1526.31
  5065.4 1527.74  5091.9 1531.12  5128.9 1533.45  5168.3 1539.09  5210.5 1541.32
  5287.7 1536.54  5314.2 1536.86  5345.9  1531.8  5368.4 1535.65  5421.1 1541.28
  5504.6  1544.6  5589.6 1550.48  5715.9 1556.12  5795.6 1561.98  5866.7 1562.57
#Mann= 4 ,-1 , 0
  4188.3     .16       0  4906.7     .07       0  5028.4     .16       0
  5866.7      .1       0
#XS Ineff= 1 ,-1
 5214.06  5512.5 1541.21
Permanent Ineff=
       T
Bank Sta=4906.7,5028.4
XS Rating Curve= 0 ,0
Exp/Cntr=0.3,0.1

Type RM Length L Ch R = 1 ,24801   ,492,492,492
BEGIN DESCRIPTION:
SOUTH GRAPE CREEK 37.0
END DESCRIPTION:
XS GIS Cut Line= 2
       2798280.7     10035273.71      2798150.58     10033597.65
#Sta/Elev= 30
  4137.5 1552.06  4231.9 1551.28  4359.7 1547.91  4371.6 1547.41  4608.9 1543.88
  4804.1 1544.05  4869.7  1544.6  4903.1 1543.53  4929.9 1542.15  4949.9 1539.18
  4959.9 1535.71    4970 1530.43    4980 1523.25    4990  1518.4  5002.1 1515.91
  5002.6  1515.8  5005.4  1515.3  5008.6  1515.8  5030.2 1517.78  5070.3 1518.67
  5101.1 1524.25  5180.6 1530.29  5265.2 1537.15    5321 1544.31  5337.4 1544.27
  5491.5 1546.21  5611.9 1549.87  5712.2 1555.59  5752.3 1560.44  5818.6 1562.53
#Mann= 10 ,-1 , 0
  4137.5     .05       0  4359.7      .1       0  4371.6     .05       0
  4804.1      .1       0  4903.1     .16       0  5002.1     .12       0
  5002.6     .07       0  5008.6     .12       0  5101.1     .16       0
  5337.4      .1       0
Bank Sta=4970,5180.6
XS Rating Curve= 0 ,0
Exp/Cntr=0.3,0.1

Type RM Length L Ch R = 1 ,24309   ,377,377,377
BEGIN DESCRIPTION:
SOUTH GRAPE CREEK 36.0
END DESCRIPTION:
XS GIS Cut Line= 2
      2798832.79     10034929.98      2798483.83     10033544.55
#Sta/Elev= 30
  4302.5  1550.1  4367.1 1549.39    4493 1545.66  4625.4 1541.68  4712.5 1541.06
  4753.8 1541.61  4783.3 1538.56  4814.2 1539.02  4830.8 1534.62  4877.1 1535.05
  4927.7  1524.9  4948.3 1520.29  4979.2 1516.28  5010.2 1515.94  5030.8 1519.37
  5049.9 1515.82  5058.7 1515.28  5061.5 1514.78  5064.7 1515.28  5072.1 1516.29
  5077.4 1522.17    5103 1526.22  5118.5  1530.7  5202.3 1542.03  5370.7 1543.06
  5626.8 1545.05  5635.5 1545.59  5688.7 1555.06  5701.1 1559.86  5731.2 1563.47
#Mann= 11 ,-1 , 0
  4302.5     .05       0  4367.1      .1       0    4493     .05       0
  4712.5      .1       0  5049.9     .16       0  5058.7     .07       0
  5064.7     .16       0  5202.3      .1       0  5370.7     .05       0
  5626.8      .1       0  5635.5     .16       0
Bank Sta=4927.7,5103
XS Rating Curve= 0 ,0
Exp/Cntr=0.3,0.1

Type RM Length L Ch R = 1 ,23932   ,697,697,697
BEGIN DESCRIPTION:
SOUTH GRAPE CREEK 35.0
END DESCRIPTION:
XS GIS Cut Line= 2
      2799171.32     10034820.54       2798770.3     10033112.28
#Sta/Elev= 30
  4304.1 1543.04  4413.8 1539.96  4619.3 1538.31  4660.3 1537.27  4685.5 1535.55
  4734.8 1533.47  4800.5 1528.63  4824.8 1527.53  4867.2 1523.57  4899.2 1517.15
  4946.9 1513.99  4978.8 1518.39    4989 1515.98  4991.5 1512.93  4994.2 1512.43
  4997.5 1512.93  5009.6  1513.5  5019.9 1516.57  5030.1  1521.3  5050.7 1523.26
  5071.2 1526.14  5079.3 1528.75  5084.5 1528.97  5091.8 1531.35  5121.7 1536.65
    5168 1542.12  5497.3 1543.31  5818.9 1546.02  6012.6 1549.88  6058.8 1551.01
#Mann= 10 ,-1 , 0
  4304.1     .05       0  4685.5     .16       0  4800.5      .1       0
  4899.2     .16       0  4991.5     .07       0  4997.5     .16       0
    5168      .1       0  5497.3     .05       0  5818.9      .1       0
  6012.6     .05       0
Bank Sta=4867.2,5050.7
XS Rating Curve= 0 ,0
Exp/Cntr=0.3,0.1

Type RM Length L Ch R = 1 ,23235   ,536,536,536
BEGIN DESCRIPTION:
SOUTH GRAPE CREEK 34.0
END DESCRIPTION:
XS GIS Cut Line= 2
      2799218.22     10034903.91      2800019.38     10033707.36
#Sta/Elev= 30
  4190.3 1545.85  4285.2 1544.42  4342.8 1541.29  4378.3 1539.06  4615.4 1535.95
  4636.5 1533.62  4659.9 1534.04  4715.4 1531.06  4795.6 1527.21  4867.6 1518.06
  4888.6 1517.62  4912.6  1513.1  4924.7  1512.8  4939.7 1514.24  4969.7 1518.71
  4993.8 1509.85  4996.6 1509.35  4999.8 1509.85  5002.4 1509.98  5020.7 1512.44
  5041.7 1520.57  5060.6 1530.22    5069 1534.42  5077.8 1535.08  5128.8 1531.86
  5175.7 1531.26  5236.9 1532.86  5326.8 1537.84  5475.1  1539.6  5630.3 1540.23
#Mann= 10 ,-1 , 0
  4190.3      .1       0  4342.8     .05       0  4715.4     .16       0
  4993.8     .07       0  4999.8     .16       0  5002.4      .1       0
  5060.6     .16       0  5175.7      .1       0  5326.8     .05       0
  5475.1      .1       0
Bank Sta=4969.7,5041.7
XS Rating Curve= 0 ,0
Exp/Cntr=0.3,0.1

Type RM Length L Ch R = 1 ,22699   ,485,485,485
BEGIN DESCRIPTION:
SOUTH GRAPE CREEK 33.0
END DESCRIPTION:
XS GIS Cut Line= 2
      2799632.08     10035341.16      2800359.81     10034092.78
#Sta/Elev= 30
  3985.9 1547.89  4098.7 1547.02  4149.1  1541.7  4175.7 1540.68  4193.5  1539.3
  4207.9 1538.16  4295.4 1535.99  4550.3 1535.19  4704.9  1532.9  4726.4 1529.87
  4763.6 1528.52  4855.3 1521.27  4896.8 1515.17  4908.9 1514.29  4955.2 1516.39
  4966.4 1514.81  4995.5 1507.29  4998.3 1506.79  5001.5 1507.29  5013.1 1509.95
    5020 1512.65  5041.5 1516.32  5047.8 1518.57    5071 1521.67    5106 1528.62
    5152 1528.35  5197.9 1530.16  5233.7 1530.46  5299.6 1532.34  5430.9 1538.34
#Mann= 10 ,-1 , 0
  3985.9     .05       0  4175.7      .1       0  4193.5     .05       0
  4855.3      .1       0  4966.4     .16       0  4995.5     .07       0
  5001.5     .16       0  5197.9      .1       0  5233.7     .16       0
  5299.6     .05       0
Bank Sta=4955.2,5041.5
XS Rating Curve= 0 ,0
Exp/Cntr=0.3,0.1

Type RM Length L Ch R = 1 ,22214   ,442,442,442
BEGIN DESCRIPTION:
SOUTH GRAPE CREEK 32.0
END DESCRIPTION:
XS GIS Cut Line= 3
       2800034.4     10035613.29      2800590.53     10034648.94
      2800596.45     10034388.63
#Sta/Elev= 30
  3953.4 1537.78  4057.1 1534.31  4160.7 1532.95  4292.6 1535.16  4437.7    1535
  4555.5 1531.46    4791 1528.08  4806.8 1527.02  4818.7 1523.67  4857.9 1522.47
  4945.6 1514.01  4967.7 1514.31  4973.5  1512.5  4975.6 1511.47  4989.2 1505.86
    4995 1504.13  5000.4    1504  5003.1  1503.5  5006.4    1504  5026.5 1507.54
  5032.3 1511.45  5038.1 1512.31  5071.8 1514.27  5101.8 1520.51  5125.8 1527.46
  5141.8 1532.53  5161.9 1534.74  5211.9 1536.58  5251.9 1535.95    5327 1537.39
#Mann= 6 ,-1 , 0
  3953.4     .05       0  4857.9     .16       0  4975.6     .05       0
  5000.4     .04       0  5006.4     .05       0  5125.8     .16       0
Bank Sta=4973.5,5038.1
XS Rating Curve= 0 ,0
Exp/Cntr=0.3,0.1

Type RM Length L Ch R = 1 ,21772   ,854,854,854
BEGIN DESCRIPTION:
SOUTH GRAPE CREEK 31.0
END DESCRIPTION:
XS GIS Cut Line= 3
      2800114.97     10035768.81      2800963.26     10034897.42
      2802158.37     10034554.27
#Sta/Elev= 30
  3874.7 1540.66  3977.3 1534.61    4100 1532.43  4397.1 1535.33  4453.7 1532.82
  4510.1 1522.98  4566.5 1518.53  4784.3 1520.19  4870.9 1513.93    4892 1516.39
  4928.3 1512.11  4969.9 1510.37  5016.3 1502.23  5019.1 1501.73  5022.3 1502.23
  5033.5 1507.44  5040.4 1516.34  5054.6 1522.48  5089.9 1522.56  5179.5 1514.35
  5210.7 1504.79  5221.1 1504.63  5356.3 1538.95  5387.5 1543.31  5470.8  1546.5
  5607.5 1542.18  5876.5 1545.23  6177.9 1562.93  6289.1 1570.63  6334.2 1572.36
#Mann= 10 ,-1 , 0
  3874.7      .1       0  3977.3     .05       0  4566.5     .16       0
  4784.3     .05       0  4928.3     .16       0  5016.3     .07       0
  5022.3     .16       0  5607.5     .05       0  6177.9      .1       0
  6289.1     .16       0
#XS Ineff= 1 ,-1
    5075 5311.93 1523.33
Permanent Ineff=
       T
Bank Sta=4892,5040.4
XS Rating Curve= 0 ,0
Exp/Cntr=0.3,0.1

Type RM Length L Ch R = 1 ,20918   ,704,704,704
BEGIN DESCRIPTION:
SOUTH GRAPE CREEK 30.0
END DESCRIPTION:
XS GIS Cut Line= 2
      2800294.68      10036080.7      2802264.13     10035205.39
#Sta/Elev= 30
  4208.2  1542.9  4245.8 1541.22  4412.6  1533.1  4432.8  1532.8  4557.4 1528.73
  4742.8 1527.32  4754.4 1524.57  4783.1 1524.52  4806.4 1528.24  4829.6 1525.58
  4854.2 1518.78  4882.7 1512.42  4904.8 1510.02  4928.1 1511.47  4956.8 1509.46
  4974.6 1504.66  5000.3 1501.65  5003.1 1501.15  5006.3 1501.65  5021.1 1504.97
    5044 1503.37  5055.3 1504.58  5073.1 1511.49  5119.6  1526.7  5183.2  1530.5
    5861 1535.65    6006  1540.6  6135.9 1549.74  6268.9 1560.59  6363.4 1570.21
#Mann= 12 ,-1 , 0
  4208.2     .05       0  4245.8      .1       0  4412.6     .05       0
  4432.8      .1       0  4742.8     .05       0  4854.2      .1       0
  4882.7     .16       0  5000.3     .07       0  5006.3     .16       0
  5183.2     .05       0  6135.9      .1       0  6268.9     .16       0
Bank Sta=4928.1,5073.1
XS Rating Curve= 0 ,0
Exp/Cntr=0.3,0.1

Type RM Length L Ch R = 1 ,20214   ,918,918,918
BEGIN DESCRIPTION:
SOUTH GRAPE CREEK 29.0
END DESCRIPTION:
XS GIS Cut Line= 3
      2800525.44     10036755.14      2801365.57     10036352.83
      2802293.92     10035306.22
#Sta/Elev= 30
  3912.7 1542.41  4071.6 1541.73  4281.9 1533.39  4448.2 1529.96  4524.9 1531.38
  4547.6 1529.51  4649.3 1530.75  4689.1  1529.1  4718.4 1530.69  4859.6 1525.71
  4916.4 1518.95  4937.3 1513.62  4959.1 1504.02  4991.2 1498.24    4994 1497.74
  4997.2 1498.24  5015.4 1499.65  5030.1 1503.54  5093.7 1511.84  5150.4  1512.7
  5270.7 1526.78  5340.3 1523.39  5377.3 1525.01  5398.2  1528.9  5674.1 1528.45
  5851.4  1533.6  5952.4 1539.42  6063.9 1548.56  6154.9 1558.79  6243.2 1566.19
#Mann= 8 ,-1 , 0
  3912.7     .05       0  4718.4      .1       0  4991.2     .07       0
  4997.2      .1       0  5015.4     .16       0  5340.3     .05       0
  5952.4      .1       0  6154.9     .16       0
Bank Sta=4937.3,5093.7
XS Rating Curve= 0 ,0
Exp/Cntr=0.3,0.1

Type RM Length L Ch R = 1 ,19296   ,554,554,554
BEGIN DESCRIPTION:
SOUTH GRAPE CREEK 28.0
END DESCRIPTION:
XS GIS Cut Line= 4
      2800878.92     10036871.21      2801909.84     10036749.02
      2802606.18     10036425.88      2802895.26     10036368.11
#Sta/Elev= 30
  3544.7 1533.06  3603.4 1530.63  3835.5 1527.53  4047.7 1526.43  4198.8 1528.69
  4422.7 1527.92  4713.6  1524.9  4757.7 1526.55  4779.8  1521.5  4865.5 1514.54
  4888.4 1509.29  4997.2 1494.45    5000 1493.95  5003.2 1494.45  5031.3 1497.88
  5048.2 1501.94  5088.4 1509.11  5143.6 1516.92  5209.7  1530.8  5308.9 1545.32
  5322.7    1549  5345.6 1558.31    5349 1561.72  5354.2 1561.72  5384.2 1573.53
    5414  1579.7  5475.2 1585.32    5516 1587.21  5535.7  1590.7  5645.3 1594.29
#Mann= 8 ,-1 , 0
  3544.7     .05       0  3603.4      .1       0  3835.5     .05       0
  4422.7      .1       0  4997.2     .07       0  5003.2      .1       0
  5048.2     .16       0  5384.2      .1       0
Bank Sta=4888.4,5088.4
XS Rating Curve= 0 ,0
Exp/Cntr=0.3,0.1

Type RM Length L Ch R = 1 ,18742   ,512,512,512
BEGIN DESCRIPTION:
SOUTH GRAPE CREEK 27.0
END DESCRIPTION:
XS GIS Cut Line= 2
      2800913.56     10037066.52        2803099.     10037027.29
#Sta/Elev= 30
  3373.7 1529.41  3388.7 1529.07  3693.3 1526.55  4417.5 1525.14  4593.4 1524.93
  4708.8 1526.07  4728.8 1522.11  4771.2 1519.05  4868.8 1507.53  4928.9  1506.2
  4968.7 1500.34  4988.9  1494.4  5005.9 1493.69  5008.6 1493.19  5011.9 1493.69
  5028.9 1496.61  5058.9 1508.58  5078.9 1522.02  5088.9 1538.67  5098.9    1561
  5108.9 1574.72  5118.9 1577.31  5168.9  1578.7    5187 1581.71  5328.9 1591.13
  5358.9 1597.14  5398.9 1614.73  5418.9 1620.04  5549.7 1629.55  5559.5 1631.16
#Mann= 11 ,-1 , 0
  3373.7     .05       0  3388.7      .1       0  3693.3     .05       0
  4417.5      .1       0  4593.4     .05       0  4771.2      .1       0
  4968.7     .16       0  5005.9     .07       0  5011.9     .16       0
    5187      .1       0  5549.7     .16       0
Bank Sta=4928.9,5058.9
XS Rating Curve= 0 ,0
Exp/Cntr=0.3,0.1

Type RM Length L Ch R = 1 ,18230   ,644,644,644
BEGIN DESCRIPTION:
SOUTH GRAPE CREEK 26.0
END DESCRIPTION:
XS GIS Cut Line= 3
      2800709.64     10037587.36      2802868.31     10037536.09
      2803057.61     10037411.86
#Sta/Elev= 30
  3134.2 1532.58  3253.1 1526.91  3620.1 1524.77  3649.3 1524.68    4413 1522.15
  4516.3 1521.55  4686.8 1522.01  4812.6 1508.35  4863.5 1507.15  4884.6 1502.73
  5000.6 1493.49  5003.3 1492.99  5006.6 1493.49  5010.2 1493.55  5083.6 1507.51
  5143.6    1529  5303.3 1546.46  5339.4 1558.98  5345.4 1564.27  5360.5 1567.16
  5366.5 1573.06  5375.6 1574.64  5381.6 1580.52  5432.8 1597.42  5438.8 1602.66
  5447.9 1603.36  5453.9  1608.8  5482.8 1618.38    5499 1623.96  5519.9 1628.92
#Mann= 13 ,-1 , 0
  3134.2     .05       0  3620.1      .1       0  3649.3     .05       0
    4413      .1       0  4516.3     .05       0  4686.8      .1       0
  4812.6     .16       0  4884.6      .1       0  5000.6     .07       0
  5006.6      .1       0  5010.2     .16       0  5482.8      .1       0
    5499     .16       0
Bank Sta=4863.5,5083.6
XS Rating Curve= 0 ,0
Exp/Cntr=0.3,0.1
