--- THREEMILE CREEK.prj (project) ---

Proj Title=THREEMILE CREEK Base Level Engineering
Current Plan=p01
Default Exp/Contr=0.3,0.1
English Units
Geom File=g01
Flow File=f01
Plan File=p01
Y Axis Title=Elevation
X Axis Title(PF)=Main Channel Distance
X Axis Title(XS)=Station
BEGIN DESCRIPTION:
THREEMILE CREEK
END DESCRIPTION:
DSS Export Rating Curves= 0
DSS Export Rating Curve Sorted= 0
DSS Export Volume Flow Curves= 0
DXF OffsetX= 0
DXF OffsetY= 0
DXF ScaleX= 1
DXF ScaleY= 10

--- THREEMILE CREEK.p01 (plan) ---

Plan Title=Multiple Run
Short Identifier=Multiple
Geom File=g01
Flow File=f01
Subcritical Flow
K Sum by GR= 0
Std Step Tol= 0.01
Critical Tol= 0.01
Num of Std Step Trials= 20
Max Error Tol= 0.3
Flow Tol Ratio= 0.001
Split Flow NTrial= 30
Split Flow Tol= 0.02
Split Flow Ratio= 0.02
Log Output Level= 0
Friction Slope Method= 1
Unsteady Friction Slope Method= 2
Unsteady Bridges Friction Slope Method= 1
Parabolic Critical Depth
Global Vel Dist=  1 , 1 , 1
Global Log Level= 0
CheckData=True
Encroach Param= -1, 0, 0, 0
BEGIN DESCRIPTION:
Multiple Run
END DESCRIPTION:

--- THREEMILE CREEK.f01 (steady flow) ---

Flow Title=Multiple
Program Version=4.10
Number of Profiles= 7
Profile Names=10-year,25-year,50-year,1pct_min,100-year,1pct_plu,500-year
River Rch & RM=THREEMILE CREEK,Reach-1         ,25418
    3069    4705    6200    5956    8055   10894   13661
River Rch & RM=THREEMILE CREEK,Reach-1         ,24308
    3069    4705    6200    5956    8055   10894   13661
River Rch & RM=THREEMILE CREEK,Reach-1         ,20140
    3268    5012    6606    6344    8580   11604   14545
River Rch & RM=THREEMILE CREEK,Reach-1         ,15008
    3371    5175    6824    6556    8867   11991   15043
River Rch & RM=THREEMILE CREEK,Reach-1         ,13812
    3505    5379    7092    6811    9211   12457   15614
River Rch & RM=THREEMILE CREEK,Reach-1         ,9911
    3527    5394    7095    6796    9191   12430   15498
Boundary for River Rch & Prof#=THREEMILE CREEK,Reach-1         , 1
Up Type= 0
Dn Type= 3
Dn Slope=0.01073
Boundary for River Rch & Prof#=THREEMILE CREEK,Reach-1         , 2
Up Type= 0
Dn Type= 3
Dn Slope=0.01073
Boundary for River Rch & Prof#=THREEMILE CREEK,Reach-1         , 3
Up Type= 0
Dn Type= 3
Dn Slope=0.01073
Boundary for River Rch & Prof#=THREEMILE CREEK,Reach-1         , 4
Up Type= 0
Dn Type= 3
Dn Slope=0.01073
Boundary for River Rch & Prof#=THREEMILE CREEK,Reach-1         , 5
Up Type= 0
Dn Type= 3
Dn Slope=0.01073
Boundary for River Rch & Prof#=THREEMILE CREEK,Reach-1         , 6
Up Type= 0
Dn Type= 3
Dn Slope=0.01073
Boundary for River Rch & Prof#=THREEMILE CREEK,Reach-1         , 7
Up Type= 0
Dn Type= 3
Dn Slope=0.01073
DSS Import GetInterval= 0
DSS Import GetPeak= 0
DSS Import FillOption= 0

--- THREEMILE CREEK.g01 (geometry) ---

Geom Title=Existing Conditions
Program Version=4.10

River Reach=THREEMILE CREEK ,Reach-1
Reach XY= 30
      2821488.47     10034673.73      2821429.58     10035048.53
      2821856.22     10035204.42      2821948.47     10035843.73
      2820991.63     10035744.98      2820830.34     10036238.36
      2821295.33     10036932.43      2820738.47     10037393.73
      2820490.93     10038570.25      2819710.23     10038779.22
      2820134.97     10040602.42      2819378.84     10040753.19
      2819233.28     10041566.45       2818761.2      10041914.8
      2818782.79     10042776.13      2818229.99     10043228.98
      2818351.05     10044446.62       2819051.7     10044916.94
      2819188.71     10045350.01      2818518.98     10046883.09
      2818973.11     10047886.36      2818563.96     10048142.21
      2817887.76     10047693.96      2817609.56     10047983.84
      2817861.32     10049262.55      2818295.39     10049884.94
      2818238.77     10050835.63      2818736.29      10051209.4
      2818082.76     10051472.85      2818106.72     10051851.62

Type RM Length L Ch R = 1 ,25418   ,1110,1110,1110
BEGIN DESCRIPTION:
THREEMILE CREEK 43.0
END DESCRIPTION:
XS GIS Cut Line= 5
      2820149.18      10034671.8       2821272.1     10034687.93
      2821627.05     10034813.78      2822188.53      10035020.3
      2823079.14     10034891.23
#Sta/Elev= 30
  3668.5 1631.75  3785.6 1621.85  3837.8 1617.61  4227.8 1583.49  4247.8 1584.27
  4297.8 1580.46  4417.9 1575.82  4607.9  1571.8  4697.9 1570.65  4861.9 1572.59
    4917 1571.47  4936.2 1570.72  4989.3 1563.59    4996 1563.54  4998.7 1563.04
    5002 1563.54  5010.5  1565.3  5166.2 1571.78  5331.1 1568.31  5478.6 1567.54
  5558.8 1570.49  5723.7    1570  5887.6 1572.06    5928 1577.83  5958.3 1585.28
  6018.9 1591.12  6291.8 1602.62    6504 1607.26    6643 1612.09  6666.3 1612.41
#Mann= 7 ,-1 , 0
  3668.5     .05       0  3785.6      .1       0  3837.8     .16       0
  4989.3     .07       0  5010.5     .16       0    6504     .05       0
    6643      .1       0
#XS Ineff= 2 ,-1
 4358.02  4853.7  1572.9 5173.26 5993.53 1571.94
Permanent Ineff=
       T       T
Bank Sta=4996,5002
XS Rating Curve= 0 ,0
Exp/Cntr=0.3,0.1

Type RM Length L Ch R = 1 ,24308   ,1785,1785,1785
BEGIN DESCRIPTION:
THREEMILE CREEK 43.0
END DESCRIPTION:
XS GIS Cut Line= 3
      2820139.57     10035113.41      2821764.58     10035571.75
      2823181.28      10035189.8
#Sta/Elev= 30
  3078.4 1621.23  3201.9 1610.63  3286.2 1596.97  3354.2 1589.66  3573.8 1573.43
  3837.8 1567.33  4116.3 1568.08  4535.9    1559  4603.9 1563.08  4682.3 1562.09
  4782.4 1564.81  4884.8 1564.32  4915.8 1561.54  4971.6 1558.72  4988.3 1557.73
  4998.4  1556.1  5011.6 1560.18  5019.4 1566.56  5046.3 1576.74  5081.1 1583.51
  5160.9 1588.11  5331.5 1590.37  5568.3 1584.75  5624.4 1587.98  5659.2  1586.3
  5773.8 1592.98  5848.4    1593  5995.3  1598.8  6233.1 1604.91  6234.1 1604.91
#Mann= 7 ,-1 , 0
  3078.4     .16       0  4971.6     .07       0  4988.3     .16       0
  5331.5      .1       0  5848.4     .05       0  5995.3      .1       0
  6233.1     .05       0
#XS Ineff= 2 ,-1
 3658.79 4075.94 1568.52 4192.95 4841.57 1564.41
Permanent Ineff=
       T       T
Bank Sta=4915.8,5011.6
XS Rating Curve= 0 ,0
Exp/Cntr=0.3,0.1

Type RM Length L Ch R = 1 ,22523   ,912,912,912
BEGIN DESCRIPTION:
THREEMILE CREEK 42.0
END DESCRIPTION:
XS GIS Cut Line= 3
      2820070.18     10035613.43      2821681.25     10036217.58
      2823013.99      10036120.4
#Sta/Elev= 30
  4070.6 1640.71  4115.5 1636.62  4218.3  1617.6  4346.9 1606.48  4432.3 1592.54
  4482.2 1581.33    4636 1568.25  4884.5 1558.71  4909.4 1552.49  4914.7 1554.95
  4923.2 1551.82  4933.8 1551.56  4939.6 1554.63    4945 1551.91  4955.2 1553.93
  4994.6 1546.66  5008.6 1548.76  5030.4 1547.97    5062 1553.14  5104.7 1556.69
    5297 1559.36  5397.1  1558.5  5467.8  1561.7  5489.2 1563.72  6039.1 1572.56
  6269.7 1578.68    6761 1601.54  6891.3 1604.78  7021.7 1612.41  7127.5 1615.11
#Mann= 5 ,-1 , 0
  4070.6      .1       0    4636     .16       0  5008.6     .07       0
  5030.4     .16       0  5467.8      .1       0
Bank Sta=4955.2,5062
XS Rating Curve= 0 ,0
Exp/Cntr=0.3,0.1

Type RM Length L Ch R = 1 ,21611   ,593,593,593
BEGIN DESCRIPTION:
THREEMILE CREEK 41.0
END DESCRIPTION:
XS GIS Cut Line= 3
      2820014.56     10036009.23      2821021.53     10036634.25
      2822895.01       10036322.
#Sta/Elev= 30
    3548 1637.72  3583.5 1633.86    3626 1622.48  3670.3 1619.51    3815 1603.49
  3851.6 1597.71  3888.2 1587.61  3924.8 1577.23  3961.4 1570.68  4070.5 1562.78
  4156.3 1559.15  4329.9 1555.64  4586.2 1555.92  4841.6 1553.51  4887.8  1550.8
  4973.4 1544.26  5000.8 1538.84  5003.5 1538.34  5006.8 1538.84  5034.2 1550.27
  5044.3 1552.63  5054.5 1552.36  5131.1 1560.14  5182.7 1560.84  5429.6 1563.49
  5885.8 1575.01  6058.1 1583.99  6078.4 1583.45  6474.4 1598.54  6632.5 1602.83
#Mann= 5 ,-1 , 0
    3548      .1       0  3888.2     .16       0  5000.8     .07       0
  5006.8     .16       0  5182.7      .1       0
Bank Sta=4887.8,5044.3
XS Rating Curve= 0 ,0
Exp/Cntr=0.3,0.1

Type RM Length L Ch R = 1 ,21018   ,269,269,269
BEGIN DESCRIPTION:
THREEMILE CREEK 40.0
END DESCRIPTION:
XS GIS Cut Line= 3
      2819945.12     10036148.12       2821299.3     10037231.47
       2822684.1     10037595.31
#Sta/Elev= 30
  3473.9 1625.75  3494.1 1622.43  3622.2 1613.92  3708.6 1601.22  3785.5 1594.01
  3843.1 1587.42  3871.9 1578.18  3913.6 1570.41  3977.6  1563.2    4056  1559.2
  4248.1 1554.07  4718.7 1551.63  4902.8 1548.47  4952.4 1541.82  4989.3 1540.48
  4992.7 1537.11  4995.4 1536.61  5010.1 1540.24  5024.5 1548.89  5030.9 1556.13
  5045.3 1560.37  5286.6 1564.65  5693.2  1570.8  5806.9 1575.06  5889.6 1575.89
    5962 1579.71  6210.2 1585.92    6339 1592.32  6582.7 1600.37  6639.9 1601.67
#Mann= 6 ,-1 , 0
  3473.9      .1       0  3785.5     .16       0  4992.7     .07       0
  5024.5     .16       0  5286.6     .05       0  6582.7      .1       0
Bank Sta=4902.8,5024.5
XS Rating Curve= 0 ,0
Exp/Cntr=0.3,0.1

Type RM Length L Ch R = 1 ,20749   ,609,609,609
BEGIN DESCRIPTION:
THREEMILE CREEK 39.0
END DESCRIPTION:
XS GIS Cut Line= 3
      2819931.23     10036502.29       2821174.3     10037453.69
      2822570.11     10037821.74
#Sta/Elev= 30
  3752.4 1601.33    3809  1600.1  3987.6 1589.32  4014.7 1585.57  4051.2 1574.86
  4072.8 1569.49  4108.2 1564.85  4236.9 1556.23  4693.4 1549.52  4735.6 1547.24
  4750.1 1548.93  4864.4 1548.44  4920.5 1545.98  4943.3 1543.92  4975.6 1536.64
  4978.4 1536.14  4981.6 1536.64  5034.8 1541.25  5057.5  1546.1  5092.9 1549.46
  5248.8 1553.08  5418.2 1559.88  5493.6 1563.47  5574.2 1563.89  6066.7 1576.83
  6149.4 1581.09  6449.3 1589.24  6563.1 1596.31    6615 1597.19  6761.3  1600.9
#Mann= 6 ,-1 , 0
  3752.4      .1       0  4051.2     .16       0  4975.6     .07       0
  4981.6     .16       0  5418.2     .05       0    6615      .1       0
Bank Sta=4920.5,5057.5
XS Rating Curve= 0 ,0
Exp/Cntr=0.3,0.1

Type RM Length L Ch R = 1 ,20140   ,299,299,299
BEGIN DESCRIPTION:
THREEMILE CREEK 38.0
END DESCRIPTION:
XS GIS Cut Line= 3
      2819368.75     10037064.81      2820875.69     10037863.42
      2822542.38     10038023.14
#Sta/Elev= 30
    3585 1587.76  3631.1 1585.77  3716.5  1582.5  3787.9 1581.29  3922.6 1577.85
  3954.5 1574.37  4004.1 1575.44  4108.3 1571.52  4250.1 1564.69  4322.1 1561.92
    4559 1553.32  4810.2  1547.6    4850 1540.69  4899.6 1536.72  4976.3 1537.39
  4995.3  1532.5    4998    1532  5001.3  1532.5  5025.9 1541.96  5042.3 1545.05
    5092 1545.72  5225.9 1546.29  5475.3 1547.27  5604.7 1558.34  5738.7  1560.3
  6056.7 1568.05  6538.9 1586.82  6680.5  1590.4  6890.9 1598.52  6964.8 1600.89
#Mann= 17 ,-1 , 0
    3585     .05       0  3631.1      .1       0  3716.5     .05       0
  3787.9      .1       0  3922.6     .05       0  4108.3      .1       0
  4250.1     .05       0  4322.1      .1       0  4810.2     .16       0
  4995.3     .07       0  5001.3     .16       0    5092      .1       0
  5225.9     .05       0  5475.3      .1       0  5738.7     .05       0
  6680.5      .1       0  6890.9     .05       0
Bank Sta=4850,5025.9
XS Rating Curve= 0 ,0
Exp/Cntr=0.3,0.1

Type RM Length L Ch R = 1 ,19841   ,589,589,589
BEGIN DESCRIPTION:
THREEMILE CREEK 37.0
END DESCRIPTION:
XS GIS Cut Line= 3
      2819347.95     10037460.65      2820806.25     10038141.19
      2822313.23     10038162.03
#Sta/Elev= 30
  3742.1 1578.31  3862.8 1575.43  4029.6 1574.62  4062.7 1572.89    4137 1573.82
  4292.5 1568.44    4468 1556.25  4542.1    1553  4691.7 1548.24  4901.6 1545.38
  4912.4 1544.85  4934.5 1538.93  4941.8 1534.42  4947.3 1535.26  4956.6 1532.38
    4990 1530.22  4992.8 1529.72    4996 1530.22  5022.8 1535.45  5068.1 1538.44
  5181.4 1543.46  5237.1 1543.03  5373.6 1543.23  5693.6  1557.5  5813.6 1558.43
  6183.7  1566.8  6233.7 1569.88  6363.7 1573.12  6683.7 1586.48  6858.5 1591.73
#Mann= 7 ,-1 , 0
  3742.1      .1       0  3862.8     .05       0  4292.5      .1       0
    4990     .07       0    4996      .1       0  5068.1     .16       0
  5237.1      .1       0
Bank Sta=4934.5,5068.1
XS Rating Curve= 0 ,0
Exp/Cntr=0.3,0.1

Type RM Length L Ch R = 1 ,19252   ,880,880,880
BEGIN DESCRIPTION:
THREEMILE CREEK 36.0
END DESCRIPTION:
XS GIS Cut Line= 3
      2818639.62     10037877.32       2820736.8     10038634.25
      2822243.59     10038516.21
#Sta/Elev= 30
  3017.6 1583.56  3417.9 1573.04  3700.7  1567.3  3908.6 1558.28  4219.8 1549.07
  4578.4 1540.27  4609.1 1537.14  4614.4 1532.98  4639.7 1534.49  4653.6 1532.58
  4670.4 1536.71  4874.5 1535.43    4896 1534.18  4983.2 1531.27  4994.2 1527.03
    4997 1526.53  5000.2 1527.03  5015.1 1531.32  5022.6  1535.8  5036.3 1539.97
  5071.7 1541.17  5253.8 1542.94  5400.1 1543.25  5670.2 1548.21  5730.3 1553.12
  6231.9 1566.19  6302.1  1570.4  6352.2 1570.57  6412.4 1574.61  6758.6 1586.73
#Mann= 10 ,-1 , 0
  3017.6     .05       0  3417.9      .1       0  3908.6     .05       0
  4219.8      .1       0    4896     .05       0  4994.2    .035       0
  5000.2     .05       0  5071.7      .1       0  5253.8     .05       0
  5400.1      .1       0
Bank Sta=4874.5,5022.6
XS Rating Curve= 0 ,0
Exp/Cntr=0.3,0.1

Type RM Length L Ch R = 1 ,18372   ,561,561,561
BEGIN DESCRIPTION:
THREEMILE CREEK 35.0
END DESCRIPTION:
XS GIS Cut Line= 3
      2818486.84     10038210.65      2820042.36     10038863.42
      2822000.73     10038891.19
#Sta/Elev= 30
    3659 1589.69  3877.9 1582.01  4166.2 1573.74  4286.9 1570.76  4471.2 1565.36
  4586.2 1560.92  4686.7 1552.92  4863.9 1543.81  4940.5 1541.81  4975.2 1538.55
  4983.8 1531.05    4996 1522.46  4998.7 1521.96    5002 1522.46  5022.8 1526.21
  5099.5 1530.24  5153.8 1533.25  5419.3 1537.69  5466.1 1537.64  5632.1 1534.96
  5850.6  1536.7  5980.2 1537.43  6069.8 1538.91  6442.2 1545.15  6502.2 1549.72
  6942.2 1562.13  7012.2 1562.14  7072.2 1565.42    7134 1565.49  7304.5 1571.91
#Mann= 13 ,-1 , 0
    3659      .1       0  3877.9     .05       0  4166.2      .1       0
  4286.9     .05       0  4471.2      .1       0    4996     .07       0
    5002      .1       0  5153.8     .05       0  5419.3      .1       0
  5466.1     .05       0  5850.6      .1       0  5980.2     .05       0
  6069.8      .1       0
Bank Sta=4983.8,5099.5
XS Rating Curve= 0 ,0
Exp/Cntr=0.3,0.1

Type RM Length L Ch R = 1 ,17811   ,626,626,626
BEGIN DESCRIPTION:
THREEMILE CREEK 34.0
END DESCRIPTION:
XS GIS Cut Line= 4
      2818486.79     10038557.85      2819618.75     10039287.03
      2820521.53     10039245.36      2822243.61     10038905.11
#Sta/Elev= 30
  3535.6 1580.84  3619.8 1577.62    3918 1568.71  4149.8 1563.68  4260.7 1562.06
  4444.6 1559.49  4444.7 1559.49  4683.8 1555.54  4865.3 1543.69  4891.8 1545.06
  4921.8 1538.42  4941.9 1527.82  4951.9 1524.65  5008.9 1519.36  5011.7 1518.86
  5014.9 1519.36    5042 1522.26    5052 1527.15  5064.5 1531.35  5123.2 1533.46
  5642.6 1529.41  5802.2 1531.64  6136.2 1538.09  6237.7 1540.27  6730.7 1553.85
  6781.6 1557.13  7097.6 1563.14  7320.3 1572.44  7454.8 1575.16  7541.2 1576.12
#Mann= 15 ,-1 , 0
  3535.6      .1       0  3619.8     .05       0    3918      .1       0
  4149.8     .05       0  4260.7      .1       0  4444.6     .05       0
  4444.7      .1       0  5008.9     .07       0  5014.9      .1       0
  5123.2     .05       0  5802.2      .1       0  6136.2     .05       0
  6237.7      .1       0  7320.3     .05       0  7454.8     .16       0
Bank Sta=4941.9,5052
XS Rating Curve= 0 ,0
Exp/Cntr=0.3,0.1

Type RM Length L Ch R = 1 ,17185   ,701,701,701
BEGIN DESCRIPTION:
THREEMILE CREEK 33.0
END DESCRIPTION:
XS GIS Cut Line= 4
       2819042.4     10039356.51      2819653.47     10039905.08
      2820340.97     10039787.03      2821500.68     10039182.87
#Sta/Elev= 30
    3905 1556.79  4048.7 1552.73  4225.8 1550.45  4494.9  1549.8  4760.2 1534.84
  4945.2 1530.51  4974.8 1526.52  4997.1 1514.89  4999.9 1514.39  5003.1 1514.89
  5078.7 1523.01    5127 1525.38  5253.8  1530.2  5390.8 1531.03    5410 1529.84
  5499.9 1527.37  5698.1 1529.38  5731.8 1528.92  6041.1 1528.84  6085.8 1531.19
  6116.6 1538.48  6142.6 1540.99  6202.5 1542.82  6225.8  1543.3  6290.3  1544.1
  6345.3 1546.79  6424.5 1546.74    6594 1550.78  6616.1 1549.97  6731.4 1554.03
#Mann= 11 ,-1 , 0
    3905      .1       0  4997.1     .07       0  5003.1      .1       0
  5078.7     .05       0  5253.8      .1       0    5410     .05       0
  5698.1      .1       0  5731.8     .05       0  6116.6      .1       0
  6202.5     .05       0  6225.8      .1       0
Bank Sta=4974.8,5127
XS Rating Curve= 0 ,0
Exp/Cntr=0.3,0.1

Type RM Length L Ch R = 1 ,16484   ,304,304,304
BEGIN DESCRIPTION:
THREEMILE CREEK 32.0
END DESCRIPTION:
XS GIS Cut Line= 3
      2819264.56     10039793.96      2820354.86     10040530.08
      2821645.03     10040807.54
#Sta/Elev= 30
  3916.8 1544.16  4063.6 1547.34  4124.1  1547.1  4199.2 1545.83    4460 1533.89
  4777.6 1526.54  4862.6  1521.5  4927.6 1520.55  4963.5 1517.62  4990.5 1508.83
  4993.2 1508.33  4996.5 1508.83  5007.4 1510.33  5029.4 1520.06  5050.4 1523.42
  5101.4  1521.8  5153.8 1523.64  5236.7 1523.36  5272.6 1525.37  5542.6 1524.85
  5790.4 1527.72  6146.4 1534.09  6258.9 1541.69  6273.3    1545  6279.3 1547.88
  6290.4 1549.33  6330.5 1549.82    6427 1554.99    6551 1560.62    6552 1560.69
#Mann= 11 ,-1 , 0
  3916.8      .1       0  4063.6     .16       0  4124.1      .1       0
  4990.5     .07       0  4996.5      .1       0  5153.8     .05       0
  5542.6      .1       0  5790.4     .05       0  6290.4      .1       0
    6427     .05       0    6551      .1       0
Bank Sta=4927.6,5029.4
XS Rating Curve= 0 ,0
Exp/Cntr=0.3,0.1

Type RM Length L Ch R = 1 ,16180   ,404,404,404
BEGIN DESCRIPTION:
THREEMILE CREEK 31.0
END DESCRIPTION:
XS GIS Cut Line= 3
      2819410.43     10039960.65      2820264.58     10040884.25
      2821459.05     10041405.09
#Sta/Elev= 30
  4043.4 1546.28  4129.3 1544.99  4213.9 1541.32  4454.8 1536.58  4660.1 1525.85
  4780.3  1523.8    4837 1519.03  4930.3 1518.67  4971.4 1515.88  4996.7 1506.62
  4999.5 1506.12  5002.7 1506.62  5028.1 1515.57  5034.9  1520.6  5041.9 1523.72
    5249 1519.47  5282.7 1518.52  5458.6 1521.29  5510.1 1522.73  5632.7 1522.94
  5760.7 1527.68  5789.6 1527.45  5841.8 1530.95  6016.7 1538.44  6115.8 1541.97
  6139.2 1541.68  6243.9  1546.8  6331.1 1549.15  6407.5 1553.66  6604.5 1559.95
#Mann= 6 ,-1 , 0
  4043.4      .1       0  4930.3     .05       0  4996.7    .035       0
  5002.7     .05       0    5249      .1       0  5458.6     .05       0
Bank Sta=4971.4,5028.1
XS Rating Curve= 0 ,0
Exp/Cntr=0.3,0.1

Type RM Length L Ch R = 1 ,15776   ,768,768,768
BEGIN DESCRIPTION:
THREEMILE CREEK 30.0
END DESCRIPTION:
XS GIS Cut Line= 3
      2819403.46     10040043.94       2819799.3     10041037.03
      2821070.12     10041787.02
#Sta/Elev= 30
  4268.1 1544.27  4510.6 1535.91  4569.9 1536.53    4720 1532.43  4817.2 1522.65
  4881.5 1520.93  4917.7 1517.75    4942 1512.44  4971.7 1511.55  4990.2 1506.86
  4998.3 1503.36  5001.1 1502.86  5004.3 1503.36  5020.2 1509.74  5032.2 1511.66
  5109.1 1522.04  5300.9  1517.2  5399.8 1515.48  5559.6 1517.52  5671.3 1517.86
  5889.6 1513.65  5983.5 1517.66  6108.1 1520.23  6305.2 1527.65  6545.2 1538.75
  6597.9 1543.91  6693.5 1547.85  6718.8 1547.32  6783.8 1549.75  6812.8 1551.16
#Mann= 11 ,-1 , 0
  4268.1      .1       0  4817.2     .16       0  4990.2     .05       0
  4998.3    .035       0  5004.3     .05       0  5300.9     .16       0
  5559.6      .1       0  5671.3     .16       0  5983.5     .05       0
  6718.8      .1       0  6783.8     .05       0
Bank Sta=4971.7,5032.2
XS Rating Curve= 0 ,0
Exp/Cntr=0.3,0.1

Type RM Length L Ch R = 1 ,15008   ,238,238,238
BEGIN DESCRIPTION:
THREEMILE CREEK 29.0
END DESCRIPTION:
XS GIS Cut Line= 2
      2818118.76     10040662.03      2820944.29     10041883.88
#Sta/Elev= 30
  3729.1 1558.85  3830.2 1555.15  4304.9 1537.26  4415.2 1531.92  4602.5 1528.19
  4651.2 1522.73  4698.7 1521.36  4804.2 1516.16  4877.7 1513.75  4909.7  1513.8
  4931.4 1513.58    4949 1508.61  4970.8 1503.99  4998.9  1502.5  5001.6    1502
  5004.9  1502.5  5015.2 1505.17  5030.8 1508.68  5120.8 1512.82  5152.9 1512.98
  5226.3 1509.99  5258.6 1509.61  5331.8 1516.59  5428.1 1516.47  5570.5 1515.17
  5859.4  1512.2  5964.9  1515.3  6467.9 1527.58  6725.3 1543.05  6807.5 1545.62
#Mann= 20 ,-1 , 0
  3729.1      .1       0  3830.2     .05       0  4304.9      .1       0
  4602.5     .05       0  4698.7     .16       0  4804.2      .1       0
  4877.7     .16       0  4909.7     .05       0  4998.9    .035       0
  5004.9     .05       0  5015.2      .1       0  5120.8     .05       0
  5152.9      .1       0  5226.3     .05       0  5331.8      .1       0
  5428.1     .05       0  5570.5      .1       0  5859.4     .16       0
  5964.9     .05       0  6725.3      .1       0
Bank Sta=4949,5030.8
XS Rating Curve= 0 ,0
Exp/Cntr=0.3,0.1

Type RM Length L Ch R = 1 ,14770   ,557,557,557
BEGIN DESCRIPTION:
THREEMILE CREEK 28.0
END DESCRIPTION:
XS GIS Cut Line= 2
      2818049.32      10040953.7      2820778.45     10041974.52
#Sta/Elev= 30
  3740.6 1556.87  3793.1  1555.8  3825.1 1553.27  3963.9 1549.95  4097.4  1544.2
  4214.1 1541.74  4580.3 1529.13  4665.6 1519.05  4764.6 1513.23  4863.9 1510.73
  4952.6 1510.38  4960.2 1508.25  4967.5 1505.61  4996.5 1498.67  4999.3 1498.17
  5002.5 1498.67  5007.9 1500.92  5031.6 1505.59  5063.8 1506.41  5148.6 1505.01
  5184.3 1506.04  5223.7  1512.2  5245.1  1513.9  5672.4 1513.18  5727.7 1510.94
  5800.3 1510.18  5838.2 1513.55  6069.8 1516.07  6344.8 1522.75  6654.4 1538.74
#Mann= 8 ,-1 , 0
  3740.6      .1       0  4214.1     .05       0  4665.6      .1       0
  4863.9     .16       0  4960.2      .1       0  4996.5     .07       0
  5002.5      .1       0  5063.8     .05       0
Bank Sta=4967.5,5031.6
XS Rating Curve= 0 ,0
Exp/Cntr=0.3,0.1

Type RM Length L Ch R = 1 ,14213   ,401,401,401
BEGIN DESCRIPTION:
THREEMILE CREEK 27.0
END DESCRIPTION:
XS GIS Cut Line= 3
      2818049.27     10041127.28      2818771.53     10041696.75
      2820712.77     10042098.86
#Sta/Elev= 30
  3899.4 1554.49  4323.3 1540.34  4344.1 1540.95    4373 1538.72    4473 1534.52
  4590.6 1528.23    4641 1525.38  4743.4 1519.87  4831.1 1511.44  4887.5 1504.18
  4938.6 1500.75  4980.7 1499.75  4989.6 1497.93  4996.8  1494.7  4999.6  1494.2
  5002.8  1494.7  5020.3 1499.77  5025.8 1504.47  5030.9 1506.44  5050.9 1508.17
  5126.1 1509.94  5729.8 1510.47  5829.7 1508.56  5898.5 1510.43  5929.2 1512.45
  6209.7  1516.2  6555.8  1524.2  6633.8 1528.13  6684.9 1529.29  6801.6 1535.96
#Mann= 9 ,-1 , 0
  3899.4     .05       0    4473      .1       0  4590.6     .05       0
    4641      .1       0  4831.1     .05       0  4996.8    .035       0
  5002.8     .05       0  5729.8      .1       0  5829.7     .05       0
Bank Sta=4887.5,5025.8
XS Rating Curve= 0 ,0
Exp/Cntr=0.3,0.1

Type RM Length L Ch R = 1 ,13812   ,519,519,519
BEGIN DESCRIPTION:
THREEMILE CREEK 26.0
END DESCRIPTION:
XS GIS Cut Line= 3
      2817743.72     10041710.63      2818618.75     10042030.08
      2820431.27     10042175.92
#Sta/Elev= 30
    3925 1556.07  3977.9 1555.26  4174.9 1546.53    4537 1524.65  4643.2 1520.55
  4679.1 1517.88  4854.6 1513.69  4946.5 1513.61  4956.6  1512.4    4963 1508.33
    4968 1511.12  4976.6 1504.83  4986.7 1496.56  4993.7 1492.77  4996.4 1492.27
  4999.7 1492.77  5035.4 1499.34  5076.9 1503.19  5157.2 1506.24  5286.5 1506.87
  5638.8 1510.36  5753.8  1507.6  5799.3 1505.89  5849.4 1510.09  5876.4 1510.58
  5963.3 1510.31  6140.4 1513.24  6280.8 1520.74  6421.3 1520.42  6674.9 1525.35
#Mann= 7 ,-1 , 0
    3925     .05       0  4993.7    .035       0  4999.7     .05       0
  5035.4      .1       0  5286.5     .05       0  5753.8      .1       0
  5876.4     .05       0
Bank Sta=4976.6,5076.9
XS Rating Curve= 0 ,0
Exp/Cntr=0.3,0.1

Type RM Length L Ch R = 1 ,13293   ,394,394,394
BEGIN DESCRIPTION:
THREEMILE CREEK 25.0
END DESCRIPTION:
XS GIS Cut Line= 2
      2817757.67     10041946.77      2819889.58     10042967.58
#Sta/Elev= 30
  3748.5 1554.07  4054.2 1535.54  4414.6 1509.94  4495.9 1506.96  4743.7 1505.12
  4850.9 1504.78  4924.6 1501.44  4932.1 1500.05  4997.1 1490.01  4999.8 1489.51
  5003.1 1490.01  5013.3 1494.74  5045.4 1501.47  5083.9    1504    5170 1505.93
  5254.9  1506.9  5290.5 1505.98  5327.2 1503.45    5357 1502.22  5419.1 1505.75
  5494.8 1506.75  5583.3  1508.3  5645.3 1510.29  5679.5  1512.4  5729.9 1512.26
    5810 1514.07  5838.2 1516.12  5875.1 1516.52    6025 1517.99  6112.2 1520.02
#Mann= 11 ,-1 , 0
  3748.5     .05       0  4743.7     .16       0  4850.9     .05       0
  4997.1    .035       0  5003.1     .05       0  5083.9     .16       0
    5170     .05       0  5327.2      .1       0  5494.8     .05       0
  5729.9      .1       0  5875.1     .05       0
Bank Sta=4932.1,5045.4
XS Rating Curve= 0 ,0
Exp/Cntr=0.3,0.1

Type RM Length L Ch R = 1 ,12899   ,413,413,413
BEGIN DESCRIPTION:
THREEMILE CREEK 24.0
END DESCRIPTION:
XS GIS Cut Line= 3
      2817625.66     10042002.27      2818410.42     10042682.86
      2819694.31     10043335.22
#Sta/Elev= 30
  3586.7 1558.19  3631.9  1556.7  3696.3 1552.37    3724 1552.11  3788.7  1546.6
  3880.8 1541.87    4235 1517.39  4425.9  1505.9  4543.4  1502.4  4684.6 1500.82
  4764.1 1500.84  4805.1  1501.4  4884.1 1502.61  4914.9 1499.96  4973.1  1493.2
  4992.3 1488.86  4995.1 1488.36  4998.3 1488.86  5004.7 1489.36  5034.2 1497.48
  5049.5  1500.1  5096.3 1502.96  5295.7 1504.32  5390.3  1499.7  5412.6 1500.92
  5466.6 1509.27  5501.6 1512.75  5813.2 1513.87  6004.1  1518.1  6065.6 1519.06
#Mann= 10 ,-1 , 0
  3586.7     .05       0  4543.4     .16       0  4684.6     .05       0
  4764.1     .16       0  4805.1      .1       0  4992.3     .07       0
  4998.3      .1       0  5096.3     .05       0  5466.6      .1       0
  6004.1     .05       0
Bank Sta=4914.9,5049.5
XS Rating Curve= 0 ,0
Exp/Cntr=0.3,0.1

Type RM Length L Ch R = 1 ,12486   ,466,466,466
BEGIN DESCRIPTION:
THREEMILE CREEK 23.0
END DESCRIPTION:
XS GIS Cut Line= 3
      2817868.77     10042571.77      2818625.69     10043300.92
       2819493.6     10043495.33
#Sta/Elev= 30
  4197.9 1529.75  4291.1 1523.82  4326.3 1524.62    4376  1518.3  4439.5 1514.33
    4475  1509.3    4482 1509.86  4577.5 1504.01  4591.2 1503.23  4763.4 1498.26
  4920.3 1496.07  4941.7  1494.4  4948.6 1492.79  4984.1 1491.38  4998.3 1489.02
  5030.5 1486.94  5033.3 1486.44  5036.5 1486.94  5047.7 1490.04    5076 1494.59
  5108.8 1497.77  5198.6 1498.94  5338.6 1499.32  5426.5 1499.76  5546.5 1502.84
  5783.7 1510.71  5846.1 1510.28  5938.3 1512.83  6040.8 1513.13  6138.3 1515.31
#Mann= 10 ,-1 , 0
  4197.9     .05       0  4577.5      .1       0  4591.2     .05       0
  4763.4      .1       0  5030.5     .07       0  5036.5      .1       0
  5108.8     .05       0  5198.6      .1       0  5338.6     .05       0
  5546.5      .1       0
Bank Sta=4941.7,5076
XS Rating Curve= 0 ,0
Exp/Cntr=0.3,0.1

Type RM Length L Ch R = 1 ,12020   ,399,399,399
BEGIN DESCRIPTION:
THREEMILE CREEK 22.0
END DESCRIPTION:
XS GIS Cut Line= 2
      2817604.89     10043370.36      2819431.26     10043543.97
#Sta/Elev= 30
  4331.2 1525.65  4480.7 1522.96  4519.4 1521.82  4696.4 1515.89  4907.4 1500.71
  4927.4 1498.26  4945.3 1494.41  4950.3 1495.87  4957.6 1493.75  4987.7 1483.97
  4997.8 1482.03  5004.8 1481.83  5007.6 1481.33  5010.8 1481.83  5037.9  1486.6
  5058.4 1487.97  5076.9 1490.32  5108.3 1493.72  5138.4 1495.47  5238.8 1495.83
  5339.1    1498    5490 1498.13    5551 1499.17  5620.6 1500.53  5686.8 1504.33
  5831.5 1506.89  5881.7 1509.17  5911.9 1509.02  6032.4 1512.18  6165.8 1513.72
#Mann= 8 ,-1 , 0
  4331.2     .05       0  4480.7      .1       0  4519.4     .05       0
  5004.8    .035       0  5010.8     .05       0  5076.9      .1       0
  5339.1     .05       0    5551      .1       0
Bank Sta=4957.6,5108.3
XS Rating Curve= 0 ,0
Exp/Cntr=0.3,0.1

Type RM Length L Ch R = 1 ,11621   ,361,361,361
BEGIN DESCRIPTION:
THREEMILE CREEK 21.0
END DESCRIPTION:
XS GIS Cut Line= 2
      2817688.22      10043877.3      2819431.22     10043668.98
#Sta/Elev= 30
  4247.9 1518.99  4262.4 1518.45  4362.3 1513.05  4429.4 1506.93  4462.1 1505.88
  4569.1 1499.95  4675.4 1495.77    4739 1493.24  4861.7 1494.21    4933 1492.95
  4953.1 1490.79  4961.5 1488.99  4973.3 1487.09  4983.3 1484.78  4991.3 1481.38
  5000.5 1480.01  5003.2 1479.51  5006.5 1480.01  5023.6 1483.87  5073.7 1490.15
  5078.7 1490.14  5088.2 1492.56  5134.4 1495.73  5236.1 1496.13  5446.6 1498.74
  5658.1 1503.93  5718.5 1506.97  5802.4 1508.29  5859.3 1510.77  6003.3 1512.62
#Mann= 13 ,-1 , 0
  4247.9     .05       0  4262.4      .1       0  4362.3     .05       0
  4462.1      .1       0  4675.4     .05       0  4861.7     .16       0
  4961.5      .1       0  5000.5     .07       0  5006.5      .1       0
  5088.2     .05       0  5236.1      .1       0  5802.4     .05       0
  5859.3      .1       0
Bank Sta=4953.1,5073.7
XS Rating Curve= 0 ,0
Exp/Cntr=0.3,0.1

Type RM Length L Ch R = 1 ,11260   ,457,457,457
BEGIN DESCRIPTION:
THREEMILE CREEK 20.0
END DESCRIPTION:
XS GIS Cut Line= 3
      2817764.56     10044189.81      2818660.42     10044120.36
      2819514.06     10043731.71
#Sta/Elev= 30
    4334  1515.4  4668.9 1497.27  4747.4    1495  4839.4 1489.94  4859.5 1486.97
    4870 1487.35  4879.5 1490.06  4889.6 1491.19  4909.6 1490.87  4919.7 1489.17
  4939.7 1484.75    4953 1484.54  4959.8 1484.24  4979.8 1477.52  4991.9 1477.34
  4994.6 1476.84  4997.9 1477.34  5009.9 1479.35    5030 1485.78    5050 1489.87
  5070.1 1491.67    5105 1492.44  5362.4 1495.72  5477.7 1499.27  5719.3 1503.99
  5758.4 1505.98    5840 1506.56  5922.6 1509.69  5953.9 1509.58  6170.5 1513.79
#Mann= 8 ,-1 , 0
    4334     .05       0  4747.4      .1       0    4953     .16       0
  4991.9     .07       0  4997.9     .16       0    5105      .1       0
  5758.4     .05       0  5953.9      .1       0
Bank Sta=4919.7,5050
XS Rating Curve= 0 ,0
Exp/Cntr=0.3,0.1

Type RM Length L Ch R = 1 ,10803   ,416,416,416
BEGIN DESCRIPTION:
THREEMILE CREEK 19.0
END DESCRIPTION:
XS GIS Cut Line= 3
      2817931.28     10044668.96      2818375.69     10044571.75
      2819335.09     10043963.28
#Sta/Elev= 30
  4450.5 1512.17  4588.9 1509.44  4688.6  1505.4  4764.9 1503.38  4823.6 1500.92
  4828.7 1499.77    4860 1499.55  4872.6 1499.09  4928.1 1492.56  4956.1 1485.73
  4964.5 1484.15  4985.7 1475.88    4998 1475.34  5000.7 1474.84    5004 1475.34
  5028.1 1480.02  5058.6  1481.6  5064.5 1483.78  5073.8 1484.62  5086.3 1487.35
    5110 1489.09  5189.1 1488.16  5392.4 1492.95  5434.7 1495.27  5492.4 1501.64
  5513.5  1502.7  5659.3 1505.47  5732.1 1504.38  5967.3 1506.96  6041.5 1508.52
#Mann= 6 ,-1 , 0
  4450.5      .1       0  4688.6     .05       0    4860      .1       0
    4998     .07       0    5004      .1       0  5967.3     .05       0
Bank Sta=4956.1,5073.8
XS Rating Curve= 0 ,0
Exp/Cntr=0.3,0.1

Type RM Length L Ch R = 1 ,10387   ,476,476,476
BEGIN DESCRIPTION:
THREEMILE CREEK 18.0
END DESCRIPTION:
XS GIS Cut Line= 3
      2818215.92     10044849.54      2818780.21     10044738.42
       2819424.4     10044041.31
#Sta/Elev= 30
    4366 1504.66  4429.7 1504.35  4542.6 1499.13  4582.7 1496.98  4680.1 1493.18
  4770.8  1490.9    4868 1487.24  4878.2 1486.32  4890.6 1483.21  4898.6 1482.41
  4950.1 1479.91  4971.1 1477.57  4978.5 1477.08    4997 1472.94  4999.8 1472.44
    5003 1472.94    5021 1481.35  5028.4 1483.26  5056.4 1485.99  5085.4 1487.23
  5147.2 1489.18  5275.6 1490.11  5346.5 1492.68  5396.4 1497.84  5435.6 1499.04
    5600 1501.89  5728.6  1503.9  5797.5 1506.18  5834.7  1507.3  5890.3  1508.8
#Mann= 13 ,-1 , 0
    4366      .1       0  4542.6     .05       0  4582.7      .1       0
  4770.8     .05       0  4971.1      .1       0    4997     .07       0
    5003      .1       0  5085.4     .16       0  5147.2      .1       0
  5435.6     .05       0    5600      .1       0  5797.5     .05       0
  5834.7      .1       0
Bank Sta=4898.6,5028.4
XS Rating Curve= 0 ,0
Exp/Cntr=0.3,0.1

Type RM Length L Ch R = 1 ,9911    ,633,633,633
BEGIN DESCRIPTION:
THREEMILE CREEK 17.0
END DESCRIPTION:
XS GIS Cut Line= 3
      2818306.25     10044884.25      2819000.69     10045085.64
      2819945.13     10044807.86
#Sta/Elev= 30
  4154.8 1502.62  4244.2 1500.98  4271.6  1499.3  4323.7 1492.58  4355.3 1489.62
  4427.8 1487.62  4541.9 1486.29  4825.5 1485.72  4907.2 1484.81  4927.7 1482.56
  4948.5 1478.87  4979.8 1475.48  4997.6  1471.5  5000.4    1471  5003.6  1471.5
  5012.5 1472.29  5021.5 1475.31  5059.1 1479.98  5079.2 1482.24  5125.7 1491.57
  5151.1 1494.05  5307.2 1501.92  5431.4 1506.24  5611.3 1512.59  5635.5 1513.08
  5649.3 1513.94  5667.7 1513.04  5688.6 1514.97  5743.9 1515.74  5862.3 1516.43
#Mann= 11 ,-1 , 0
  4154.8      .1       0  4541.9     .05       0  4825.5      .1       0
  4997.6     .07       0  5003.6      .1       0  5059.1     .16       0
  5307.2      .1       0  5431.4     .16       0  5611.3      .1       0
  5635.5     .05       0  5743.9      .1       0
Bank Sta=4927.7,5079.2
XS Rating Curve= 0 ,0
Exp/Cntr=0.3,0.1

Type RM Length L Ch R = 1 ,9278    ,483,483,483
BEGIN DESCRIPTION:
THREEMILE CREEK 16.0
END DESCRIPTION:
XS GIS Cut Line= 2
      2817958.99     10045078.68      2819652.46     10045939.29
#Sta/Elev= 30
  3742.9 1505.13  3856.7 1500.72  3923.5 1492.21    3968 1489.31  4028.4 1487.12
  4054.2 1486.43  4162.5 1483.87  4370.5 1482.57  4662.1 1483.49  4869.9  1480.2
  4908.1 1480.39  4920.1 1479.01  4942.6 1475.14  4980.5 1473.17  4987.4 1469.46
  4994.1 1468.17  4996.8 1467.67  5000.1 1468.17  5009.9 1469.45  5032.3 1475.04
  5041.6 1477.37  5047.2 1479.95  5054.7 1482.28  5091.7 1488.77  5108.4 1488.44
    5114 1489.71  5137.2 1490.51  5245.5 1495.41  5464.4 1502.82  5642.5 1506.12
#Mann= 9 ,-1 , 0
  3742.9      .1       0  4028.4     .16       0  4054.2      .1       0
  4162.5     .05       0  4869.9      .1       0  4994.1     .07       0
  5000.1      .1       0  5137.2     .16       0  5245.5      .1       0
Bank Sta=4920.1,5047.2
XS Rating Curve= 0 ,0
Exp/Cntr=0.3,0.1

Type RM Length L Ch R = 1 ,8795    ,579,579,579
BEGIN DESCRIPTION:
THREEMILE CREEK 15.0
END DESCRIPTION:
XS GIS Cut Line= 3
      2817764.59     10045224.54      2818625.69     10045974.53
      2819868.75      10046377.3
#Sta/Elev= 30
  3688.2 1507.95  3945.9 1499.88  4044.8 1492.37  4079.9 1491.79    4116 1485.69
  4136.9 1486.13  4151.1 1483.33  4215.7 1481.95  4417.2 1480.71  4418.6 1480.72
  4668.1 1480.85  4669.1 1480.87  4795.5 1481.43  4904.3 1479.46    4937 1479.27
  4948.7  1476.7  4974.2 1467.82  4987.7 1466.23  4990.5 1465.73  4993.7 1466.23
  5030.5 1470.91  5070.2 1477.48  5126.2 1479.93  5278.9 1484.32  5337.6 1491.61
  5411.2 1494.66  5673.6 1497.77  5927.2 1495.77  5968.3  1498.4  6136.8 1501.18
#Mann= 16 ,-1 , 0
  3688.2      .1       0  3945.9     .16       0  4215.7      .1       0
  4417.2     .05       0  4418.6      .1       0  4668.1     .05       0
  4669.1      .1       0  4795.5     .05       0  4904.3      .1       0
  4987.7     .07       0  4993.7      .1       0  5030.5     .16       0
  5126.2      .1       0  5278.9     .16       0  5673.6      .1       0
  5927.2     .05       0
Bank Sta=4948.7,5070.2
XS Rating Curve= 0 ,0
Exp/Cntr=0.3,0.1

Type RM Length L Ch R = 1 ,8216    ,431,431,431
BEGIN DESCRIPTION:
THREEMILE CREEK 14.0
END DESCRIPTION:
XS GIS Cut Line= 3
      2817459.06     10046648.14      2818472.92     10046530.08
      2819575.24      10046724.2
#Sta/Elev= 30
  3842.4 1509.91  3867.9 1509.16    3974 1505.54  4133.8 1499.43  4201.5  1495.5
  4343.2 1487.83  4395.5 1484.35  4516.3 1479.81  4536.5 1476.94  4586.4 1473.36
  4637.1 1471.19  4697.2 1475.36  4756.3 1476.85  4889.1 1477.54  4939.8 1475.18
    4973 1469.11  4980.4 1466.27  4997.7 1464.21  5000.5 1463.71  5003.7 1464.21
  5051.5  1472.9  5081.4 1475.23  5262.6 1477.63  5659.1 1481.72    5761 1481.37
    5837 1481.49  5896.3 1483.72  5934.9 1487.08  5959.9 1487.36  5982.4 1489.02
#Mann= 12 ,-1 , 0
  3842.4      .1       0  3867.9     .05       0    3974      .1       0
  4201.5     .05       0  4343.2      .1       0  4586.4     .05       0
  4756.3      .1       0  4997.7     .07       0  5003.7      .1       0
  5262.6     .05       0    5761      .1       0  5959.9     .16       0
Bank Sta=4939.8,5081.4
XS Rating Curve= 0 ,0
Exp/Cntr=0.3,0.1

Type RM Length L Ch R = 1 ,7785    ,762,762,762
BEGIN DESCRIPTION:
THREEMILE CREEK 13.0
END DESCRIPTION:
XS GIS Cut Line= 2
      2817827.08     10047037.03      2819673.84     10046863.46
#Sta/Elev= 30
  4303.3 1497.44  4372.6 1494.59  4625.6 1487.28  4767.5 1483.66  4847.1 1480.94
  4917.4 1480.55  4924.4 1480.26    4931 1478.67  4957.6 1477.03  4967.6  1474.2
  4987.7 1464.38  4997.7 1461.39  5004.8 1461.23  5007.5 1460.73  5010.8 1461.23
    5033 1466.45  5098.2 1472.13  5218.7 1472.81  5319.1  1475.5  5475.8 1474.71
  5690.8 1477.42  5901.7 1478.44  5996.1 1481.54  6030.1 1484.43  6042.3 1485.56
  6052.4 1484.63  6062.4 1485.29  6082.5 1489.71  6129.6 1493.44  6158.2 1495.43
#Mann= 10 ,-1 , 0
  4303.3      .1       0  4372.6     .05       0  4625.6      .1       0
  4767.5     .05       0    4931      .1       0  5004.8     .07       0
  5010.8      .1       0  5475.8     .05       0  6030.1     .16       0
  6129.6     .05       0
Bank Sta=4967.6,5098.2
XS Rating Curve= 0 ,0
Exp/Cntr=0.3,0.1

Type RM Length L Ch R = 1 ,7023    ,1092,1092,1092
BEGIN DESCRIPTION:
THREEMILE CREEK 12.0
END DESCRIPTION:
XS GIS Cut Line= 3
      2817945.16     10047210.65      2818695.14     10047641.19
        2819645.     10047516.39
#Sta/Elev= 30
  3933.2 1492.51    4096 1487.69  4130.7 1486.68  4259.2 1481.92  4427.8 1475.22
  4574.5 1470.91  4685.7 1469.45  4895.4 1470.86  4962.7 1467.64    5003 1457.64
  5010.1 1457.35  5012.9 1456.85  5016.1 1457.35  5047.8 1463.95  5073.6 1463.36
  5121.5 1467.54  5126.5 1466.29  5224.9 1471.93  5279.5 1470.97    5337 1471.48
  5431.3 1474.09    5467 1476.51  5487.2 1479.52    5505 1478.81  5527.8 1481.07
  5557.8 1484.33  5627.9 1487.36    5666 1490.57  5727.9 1493.65    5756 1495.47
#Mann= 14 ,-1 , 0
  3933.2     .05       0    4096      .1       0  4130.7     .05       0
  4259.2      .1       0  4427.8     .05       0  4685.7     .16       0
  5010.1     .07       0  5016.1     .16       0  5279.5     .05       0
    5337      .1       0  5527.8     .16       0  5627.9     .05       0
    5666      .1       0  5727.9     .05       0
Bank Sta=4962.7,5121.5
XS Rating Curve= 0 ,0
Exp/Cntr=0.3,0.1

Type RM Length L Ch R = 1 ,5931    ,958,958,958
BEGIN DESCRIPTION:
THREEMILE CREEK 11.0
END DESCRIPTION:
XS GIS Cut Line= 4
      2817979.86     10047280.08      2818368.75     10047800.92
      2818278.47     10048217.58      2818459.01     10048467.56
#Sta/Elev= 30
  4162.2 1490.63    4270 1487.15  4420.8 1480.37  4435.4 1478.81  4506.2 1477.34
  4535.4  1475.7  4591.7 1471.05  4614.7 1467.81  4650.1 1464.59  4700.1 1463.31
  4833.8 1466.31    4883 1465.24  4907.2 1463.39  4937.9 1459.27  4968.6 1458.21
  4976.3 1455.99  4981.4 1453.18    4986 1453.03  4988.8 1452.53    4992 1453.03
  4999.3 1453.13  5021.1  1458.2  5025.4 1461.21  5030.6 1463.27  5040.2 1465.22
  5060.7 1466.74  5238.5 1468.59  5417.9 1476.32  5471.7 1479.15  5546.9 1480.21
#Mann= 6 ,-1 , 0
  4162.2     .05       0    4270      .1       0    4986    .035       0
    4992      .1       0  5021.1      .1       0  5417.9     .05       0
Bank Sta=4907.2,5030.6
XS Rating Curve= 0 ,0
Exp/Cntr=0.3,0.1

Type RM Length L Ch R = 1 ,4973    ,577,577,577
BEGIN DESCRIPTION:
THREEMILE CREEK 10.0
END DESCRIPTION:
XS GIS Cut Line= 2
      2817292.37      10047766.2      2818444.28     10048494.82
#Sta/Elev= 30
  4619.9 1508.05  4795.8 1505.56  4868.8 1502.97    4884 1500.39  4889.9 1500.49
  4905.2 1494.78  4911.1 1494.84  4920.5 1492.03  4926.4 1491.92  4934.8 1489.02
  4941.7 1484.26  4947.6 1483.36  4956.9 1477.62  4962.8  1475.4  4970.3 1463.35
  4978.1 1454.34    4984 1451.35  4996.3 1447.44  4999.1 1446.94  5002.3 1447.44
  5035.8 1455.11  5041.7 1455.21  5087.5 1461.06    5224 1461.85  5266.3 1463.53
  5579.2 1464.97  5673.3 1467.02    5808 1473.79  5913.2 1479.12  5982.9 1479.79
#Mann= 4 ,-1 , 0
  4619.9      .1       0  4996.3     .07       0  5002.3      .1       0
    5808     .05       0
Bank Sta=4978.1,5041.7
XS Rating Curve= 0 ,0
Exp/Cntr=0.3,0.1

Type RM Length L Ch R = 1 ,4396    ,349,349,349
BEGIN DESCRIPTION:
THREEMILE CREEK 9.0
END DESCRIPTION:
XS GIS Cut Line= 2
      2817278.52     10048550.92      2818320.14     10048516.19
#Sta/Elev= 30
  4654.5 1495.93  4668.8 1495.98  4754.5 1496.72  4786.4 1495.48  4804.5 1494.05
  4824.5 1491.38  4844.6 1487.09  4860.7 1484.69  4904.6 1478.35  4944.6 1474.29
  4954.6 1472.44  4964.6 1468.33  4974.6 1461.29  4984.6 1452.42  4994.6 1446.79
  5001.6  1445.9  5004.4  1445.4  5007.6  1445.9  5014.6 1446.82  5019.9 1448.85
  5034.7 1450.93  5064.7 1453.57  5124.7 1458.56  5264.8 1462.46  5374.8 1462.57
  5434.9  1463.9  5534.9 1468.24  5620.3 1473.54    5668 1474.68  5696.7 1475.84
#Mann= 7 ,-1 , 0
  4654.5     .16       0  4668.8      .1       0  4786.4     .16       0
  4860.7      .1       0  5001.6     .07       0  5007.6      .1       0
    5668     .05       0
Bank Sta=4984.6,5064.7
XS Rating Curve= 0 ,0
Exp/Cntr=0.3,0.1

Type RM Length L Ch R = 1 ,4047    ,376,376,376
BEGIN DESCRIPTION:
THREEMILE CREEK 8.0
END DESCRIPTION:
XS GIS Cut Line= 2
      2817382.63     10048960.64      2818520.47     10048648.43
#Sta/Elev= 30
  4612.9 1490.49  4696.2 1491.75  4712.3 1492.87  4775.5 1491.05  4809.9 1488.78
  4844.4 1484.82  4849.6 1485.47    4884 1479.93    4930 1476.22  4940.4 1471.74
  4950.8 1462.42  4958.1 1454.23  4971.5  1447.9  4992.3 1445.22  4994.7 1444.02
  4997.5 1443.52  5000.7 1444.02    5013 1445.74  5044.1 1452.61  5064.8 1453.44
    5096 1456.89  5137.4 1457.79  5158.2  1459.4    5293 1461.66  5396.7 1467.42
  5452.6 1468.58  5674.9  1477.4  5742.1 1478.61  5753.6 1479.13  5792.8 1479.31
#Mann= 5 ,-1 , 0
  4612.9      .1       0  4994.7     .07       0  5000.7      .1       0
  5742.1     .05       0  5753.6      .1       0
Bank Sta=4958.1,5044.1
XS Rating Curve= 0 ,0
Exp/Cntr=0.3,0.1

Type RM Length L Ch R = 1 ,3671    ,356,356,356
BEGIN DESCRIPTION:
THREEMILE CREEK 7.0
END DESCRIPTION:
XS GIS Cut Line= 2
      2817570.16     10049231.47      2818743.62     10049189.81
#Sta/Elev= 30
  4722.2 1485.41  4760.5 1483.81  4802.5 1483.67  4900.6 1476.45  4910.6 1474.97
  4960.7 1463.03  4970.7 1458.34  4980.7 1450.98  4990.7 1444.92  5000.7 1440.72
  5007.7 1439.65  5010.4 1439.15  5013.7 1439.65  5040.7 1448.34  5060.7 1450.85
  5086.5 1451.29  5126.4 1454.35  5170.8 1455.01  5220.8 1457.44  5270.9 1457.39
  5320.9 1459.33    5431 1459.82    5511 1461.43    5551 1463.17  5631.1  1464.1
  5681.1 1466.32  5701.1 1468.25  5731.1 1468.39  5824.7 1473.07  5896.4 1476.16
#Mann= 6 ,-1 , 0
  4722.2      .1       0  5007.7     .07       0  5013.7      .1       0
  5086.5     .16       0  5126.4      .1       0  5824.7     .05       0
Bank Sta=4980.7,5060.7
XS Rating Curve= 0 ,0
Exp/Cntr=0.3,0.1

Type RM Length L Ch R = 1 ,3315    ,209,209,209
BEGIN DESCRIPTION:
THREEMILE CREEK 6.0
END DESCRIPTION:
XS GIS Cut Line= 2
      2817535.38     10049523.14      2818750.67     10049550.92
#Sta/Elev= 30
  4526.7 1477.18  4548.7 1478.43  4569.8  1478.2  4647.3 1471.12  4745.9  1464.5
  4869.9  1460.2  4889.9 1456.93  4919.9 1456.23  4943.1 1451.88  4959.9 1447.37
  4979.9 1442.76  4996.9 1442.21  4999.7 1441.71  5002.9 1442.21  5019.9 1445.33
  5049.9  1446.8  5089.9 1447.24  5140.3 1450.74    5220 1453.74  5238.9 1456.27
    5250  1457.8  5335.3 1459.36    5350 1459.85    5380 1458.37  5436.5 1462.99
    5480 1465.88  5633.2  1472.5  5680.1 1474.26  5718.9  1473.9  5742.3    1474
#Mann= 13 ,-1 , 0
  4526.7     .08       0  4548.7     .05       0  4647.3      .1       0
  4745.9     .05       0  4943.1     .16       0  4996.9     .07       0
  5002.9     .16       0  5140.3      .1       0  5238.9     .16       0
  5335.3      .1       0  5436.5     .16       0  5633.2     .05       0
  5718.9      .1       0
Bank Sta=4959.9,5049.9
XS Rating Curve= 0 ,0
Exp/Cntr=0.3,0.1

Type RM Length L Ch R = 1 ,3106    ,385,385,385
BEGIN DESCRIPTION:
Mapping XS b368eee8
END DESCRIPTION:
XS GIS Cut Line= 2
      2817646.57     10049655.09      2818799.28     10049724.53
#Sta/Elev= 30
  4496.2 1470.11  4598.6 1463.84  4708.5  1459.5  4848.7 1458.23  4908.8 1456.63
  4928.9 1454.38  4938.9 1451.79  4948.9 1445.55  4958.9 1441.06  4968.9 1441.59
    4996 1438.19  4998.8 1437.69    5002 1438.19    5019  1441.6  5039.1 1443.46
  5059.9  1443.7  5099.2 1446.65  5129.2 1452.44  5179.3 1457.99  5239.4 1459.03
  5269.5 1461.38  5359.7 1464.24  5386.5  1466.9  5391.5 1466.01  5409.7 1468.42
  5449.8 1471.51  5479.9 1470.52  5499.9  1473.6  5519.1    1474    5651 1473.62
#Mann= 5 ,-1 , 0
  4496.2     .08       0  4598.6     .05       0    4996     .04       0
    5002     .05       0  5519.1      .1       0
Bank Sta=4948.9,5099.2
XS Rating Curve= 0 ,0
Exp/Cntr=0.3,0.1

Type RM Length L Ch R = 1 ,2721    ,262,262,262
BEGIN DESCRIPTION:
THREEMILE CREEK 5.0
END DESCRIPTION:
XS GIS Cut Line= 3
      2817653.44     10049682.84      2818368.75     10050071.75
      2818757.59     10050050.92
#Sta/Elev= 30
    4322 1469.28  4380.7 1466.06    4427 1463.79  4536.7  1460.2  4604.3 1458.73
  4646.4 1458.64  4756.2  1455.9  4791.8 1453.47  4797.5 1454.86  4813.7 1452.04
  4819.4 1454.49  4827.9 1453.84  4865.9 1450.65  4944.8    1446  4966.6 1443.01
  4975.6  1439.5  4985.5 1436.45  4988.2 1435.95  4991.5 1436.45  5004.6 1436.92
  5042.6 1446.75  5051.5 1446.49  5064.5 1449.52  5070.2 1448.86  5085.4 1453.27
  5176.1 1462.49  5246.1 1468.76  5341.4 1471.26  5487.3 1472.37  5525.6 1472.98
#Mann= 17 ,-1 , 0
    4322     .08       0  4380.7     .05       0    4427     .08       0
  4536.7     .05       0  4604.3     .08       0  4646.4     .05       0
  4756.2     .16       0  4827.9     .08       0  4865.9     .05       0
  4975.6     .16       0  4985.5     .07       0  4991.5     .16       0
  5051.5     .05       0  5085.4     .16       0  5176.1      .1       0
  5341.4     .05       0  5487.3      .1       0
Bank Sta=4944.8,5042.6
XS Rating Curve= 0 ,0
Exp/Cntr=0.3,0.1

Type RM Length L Ch R = 1 ,2459    ,209,209,209
BEGIN DESCRIPTION:
Mapping XS 459550fc
END DESCRIPTION:
XS GIS Cut Line= 4
      2817639.59      10049703.7      2817972.92     10049918.97
       2818674.3     10050675.92      2818938.24     10050655.08
#Sta/Elev= 30
    4134 1469.15  4142.6 1468.78  4258.3 1464.27  4336.8 1460.66  4372.6 1459.78
  4486.9 1457.93    4531  1457.7  4670.7 1455.84    4776 1453.95    4878 1450.35
  4941.5 1445.06  4995.2 1435.79    4998 1435.29  5001.2 1435.79  5026.6  1438.4
  5032.3 1441.08  5061.7 1446.02  5075.9 1443.66  5082.7 1445.88  5089.7 1444.51
  5096.9 1447.54  5104.2 1446.17  5111.1 1448.57  5118.4 1447.23  5252.8 1458.35
    5267  1456.9    5458 1460.34  5687.3 1467.65  5755.3 1467.79  5827.5 1467.38
#Mann= 14 ,-1 , 0
    4134     .08       0  4142.6     .05       0  4258.3     .08       0
  4336.8     .05       0  4372.6     .08       0  4486.9     .05       0
    4531     .08       0  4670.7     .05       0    4776     .08       0
  4995.2     .07       0  5001.2     .08       0  5032.3     .05       0
  5089.7     .08       0  5755.3      .1       0
Bank Sta=4941.5,5061.7
XS Rating Curve= 0 ,0
Exp/Cntr=0.3,0.1

Type RM Length L Ch R = 1 ,2250    ,0,0,0
BEGIN DESCRIPTION:
THREEMILE CREEK 4.0
END DESCRIPTION:
XS GIS Cut Line= 4
      2817528.48     10049773.15      2817903.47     10050064.81
      2818570.14     10050766.19       2818874.6     10050703.92
#Sta/Elev= 30
  3970.9 1474.12  4127.9 1469.99  4235.6 1463.11    4477  1456.6  4788.4 1454.77
  4908.5  1449.9  4929.6 1446.42    4951 1445.72  4972.1 1442.52  4979.3 1441.87
  4986.2 1435.94  4997.4 1433.52  5000.1 1433.02  5003.4 1433.52  5021.8 1435.69
  5028.7 1439.65    5036 1439.67  5042.8 1442.58  5085.3 1447.95  5113.6  1448.3
    5163 1455.04  5184.4 1456.31    5326 1454.61  5413.6 1455.73    5463 1459.05
  5501.7 1459.58  5534.4 1458.84  5555.3 1463.26  5656.9 1467.12  5724.4 1467.58
#Mann= 4 ,-1 , 0
  3970.9     .05       0  4997.4     .04       0  5003.4     .05       0
  5501.7     .08       0
Bank Sta=4972.1,5042.8
XS Rating Curve= 0 ,0
Exp/Cntr=0.3,0.1

Chan Stop Cuts=-1
Use User Specified Reach Order=0
Composite Channel Slope=5
