--- UNT007 IN NNOGR.prj (project) ---

Proj Title=UNT007 IN NNOGR Base Level Engineering
Current Plan=p01
Default Exp/Contr=0.3,0.1
English Units
Geom File=g01
Flow File=f01
Plan File=p01
Y Axis Title=Elevation
X Axis Title(PF)=Main Channel Distance
X Axis Title(XS)=Station
BEGIN DESCRIPTION:
UNT007 IN NNOGR
END DESCRIPTION:
DSS Export Rating Curves= 0
DSS Export Rating Curve Sorted= 0
DSS Export Volume Flow Curves= 0
DXF OffsetX= 0
DXF OffsetY= 0
DXF ScaleX= 1
DXF ScaleY= 10

--- UNT007 IN NNOGR.p01 (plan) ---

Plan Title=Multiple Run
Short Identifier=Multiple
Geom File=g01
Flow File=f01
Subcritical Flow
K Sum by GR= 0
Std Step Tol= 0.01
Critical Tol= 0.01
Num of Std Step Trials= 20
Max Error Tol= 0.3
Flow Tol Ratio= 0.001
Split Flow NTrial= 30
Split Flow Tol= 0.02
Split Flow Ratio= 0.02
Log Output Level= 0
Friction Slope Method= 1
Unsteady Friction Slope Method= 2
Unsteady Bridges Friction Slope Method= 1
Parabolic Critical Depth
Global Vel Dist=  1 , 1 , 1
Global Log Level= 0
CheckData=True
Encroach Param= -1, 0, 0, 0
BEGIN DESCRIPTION:
Multiple Run
END DESCRIPTION:

--- UNT007 IN NNOGR.f01 (steady flow) ---

Flow Title=Multiple
Number of Profiles=7
Profile Names=10-year,25-year,50-year,1pct_min,100-year,1pct_plu,500-year
River Rch & RM= UNT007 IN NNOGR,Reach-1,21882
     847    1232    1569    1463    1978    2675    3157
River Rch & RM= UNT007 IN NNOGR,Reach-1,12903
    1053    1538    1962    1829    2474    3346    3954
Boundary for River Rch & Prof#=UNT007 IN NNOGR,Reach-1,1
Up Type=0
Dn Type=3
Dn Slope=0.005
Boundary for River Rch & Prof#=UNT007 IN NNOGR,Reach-1,2
Up Type=0
Dn Type=3
Dn Slope=0.005
Boundary for River Rch & Prof#=UNT007 IN NNOGR,Reach-1,3
Up Type=0
Dn Type=3
Dn Slope=0.005
Boundary for River Rch & Prof#=UNT007 IN NNOGR,Reach-1,4
Up Type=0
Dn Type=3
Dn Slope=0.005
Boundary for River Rch & Prof#=UNT007 IN NNOGR,Reach-1,5
Up Type=0
Dn Type=3
Dn Slope=0.005
Boundary for River Rch & Prof#=UNT007 IN NNOGR,Reach-1,6
Up Type=0
Dn Type=3
Dn Slope=0.005
Boundary for River Rch & Prof#=UNT007 IN NNOGR,Reach-1,7
Up Type=0
Dn Type=3
Dn Slope=0.005

--- UNT007 IN NNOGR.g01 (geometry) ---

Geom Title=Existing Conditions
Program Version=4.10

River Reach=UNT007 IN NNOGR ,Reach-1
Reach XY= 30
      2772433.47     10070758.73      2773297.57     10069935.34
      2773191.32     10069726.22      2773707.99      10069263.2
       2773791.4     10068394.86      2774177.57     10067913.86
      2774580.02      10067516.8      2775304.93     10067413.44
       2775966.2     10066719.16      2776278.55     10066843.68
      2776318.91      10066467.7      2776785.05     10066074.75
      2776478.71     10065598.12      2776549.24     10065252.59
      2776826.58     10065325.77      2776960.83     10064471.38
      2777757.38      10064441.1      2778465.29     10064032.49
      2778430.47     10063598.99      2778766.47     10063378.01
      2778877.47     10062793.19      2778691.14      10062544.9
      2779206.75     10061607.94      2779171.39     10060494.95
      2779658.34     10060028.69      2779893.22     10059080.74
      2780394.71      10058752.8      2779976.14     10058426.97
      2780197.15     10057295.04      2779675.37     10056465.27

Type RM Length L Ch R = 1 ,21882   ,304,304,304
BEGIN DESCRIPTION:
UNT007 IN NNOGR 44.0
END DESCRIPTION:
XS GIS Cut Line= 2
      2772632.31     10070721.33      2772344.07     10070495.61
#Sta/Elev= 30
  4856.9 1724.85  4864.6 1724.19  4879.1 1723.68  4922.5 1723.51  4928.8 1723.83
  4936.9 1723.05  4943.3 1723.12  4957.7 1722.29  4972.2 1720.48  4986.7 1716.75
    4993 1715.56  4998.1 1713.83  5000.9 1713.33  5004.1 1713.83  5007.5 1715.07
  5014.2 1715.35  5021.9 1714.81  5028.3 1716.78  5036.4 1715.54  5042.7 1717.91
  5050.8 1716.51  5057.2 1718.67    5065 1719.89  5071.7  1722.6    5078 1723.53
  5092.5 1723.49    5115 1724.15  5121.4 1723.96  5128.5  1724.4    5223    1726
#Mann= 3 ,-1 , 0
  4856.9      .1       0  4998.1     .07       0  5004.1      .1       0
Bank Sta=4998.1,5004.1
XS Rating Curve= 0 ,0
Exp/Cntr=0.3,0.1

Type RM Length L Ch R = 1 ,21578   ,392,392,392
BEGIN DESCRIPTION:
UNT007 IN NNOGR 43.0
END DESCRIPTION:
XS GIS Cut Line= 3
        2772780.     10070669.54        2772688.     10070331.04
      2772358.14     10070310.21
#Sta/Elev= 30
  4736.8 1723.42  4742.8 1722.51    4760 1721.21  4799.8 1719.57  4815.4 1719.52
  4834.4 1719.97  4874.2 1718.18  4898.3  1718.3  4919.2 1718.94  4929.4 1718.41
  4948.6 1716.28  4953.8 1716.63  4970.8 1715.02  4981.2  1713.6  4988.4 1711.05
  4998.9 1709.73  5001.6 1709.23  5004.9 1709.73  5012.3 1710.28  5022.6 1711.87
  5028.2 1714.62  5043.3 1716.65  5053.7 1717.64  5089.9 1717.85  5123.2  1718.9
  5137.2 1718.85  5282.7 1721.53  5307.6 1721.05  5327.6 1722.44  5418.1 1724.56
#Mann= 3 ,-1 , 0
  4736.8      .1       0  4998.9     .07       0  5004.9      .1       0
Bank Sta=4998.9,5004.9
XS Rating Curve= 0 ,0
Exp/Cntr=0.3,0.1

Type RM Length L Ch R = 1 ,21186   ,511,511,511
BEGIN DESCRIPTION:
UNT007 IN NNOGR 42.0
END DESCRIPTION:
XS GIS Cut Line= 4
      2773252.25      10070539.4      2773194.95     10070456.04
       2772731.4     10070145.28      2772448.45     10070232.07
#Sta/Elev= 30
  4592.6 1715.35  4627.8  1715.4  4743.2 1713.17  4773.2 1713.33  4800.3 1712.48
  4851.3 1711.88  4923.3 1711.99  4944.4  1712.5  4959.3 1712.19  4980.4 1709.27
  4995.4 1706.38  4999.5 1706.37  5002.3 1705.87  5005.5 1706.37  5010.4 1708.04
  5016.4 1708.26  5025.4 1709.66  5031.4 1709.16  5046.4 1712.01  5061.4 1712.74
  5067.4 1712.17  5133.4 1713.21  5139.4 1712.92  5154.4  1713.7  5175.5 1713.69
  5190.5 1714.32  5247.5 1714.71  5365.3 1717.71    5436  1718.8  5547.8  1721.6
#Mann= 3 ,-1 , 0
  4592.6      .1       0  4999.5     .07       0  5005.5      .1       0
Bank Sta=4999.5,5005.5
XS Rating Curve= 0 ,0
Exp/Cntr=0.3,0.1

Type RM Length L Ch R = 1 ,20675   ,699,699,699
BEGIN DESCRIPTION:
UNT007 IN NNOGR 41.0
END DESCRIPTION:
XS GIS Cut Line= 3
      2773479.64     10070221.64      2773016.13     10069890.07
      2772563.21     10070155.57
#Sta/Elev= 30
    4656 1708.63    4677 1708.82  4783.9 1706.89  4887.7 1706.17  4955.9 1706.01
  4985.4 1703.05  4997.2  1699.6  4999.9  1699.1  5003.2  1699.6    5014  1702.6
    5021 1703.77  5058.9 1704.05  5086.2 1705.88    5107 1706.38  5178.3 1706.83
    5193 1707.44  5213.9  1707.2  5248.9 1708.05  5321.9 1710.05  5404.9 1711.13
    5445 1711.27  5487.8 1712.58  5534.6 1713.44    5578 1715.03  5615.1 1713.05
  5620.9 1713.67  5636.6 1713.93  5642.4 1715.03  5663.9 1716.25  5750.9 1718.21
#Mann= 9 ,-1 , 0
    4656      .1       0  4887.7     .05       0  4997.2    .035       0
  5003.2     .05       0  5058.9      .1       0  5248.9     .05       0
  5404.9      .1       0  5487.8     .05       0  5534.6      .1       0
Bank Sta=4997.2,5003.2
XS Rating Curve= 0 ,0
Exp/Cntr=0.3,0.1

Type RM Length L Ch R = 1 ,19976   ,803,803,803
BEGIN DESCRIPTION:
UNT007 IN NNOGR 40.0
END DESCRIPTION:
XS GIS Cut Line= 3
      2773576.73     10070235.18      2773427.43     10069592.85
      2772885.79     10069155.37
#Sta/Elev= 30
  4227.5 1708.26  4243.2 1708.56  4341.9 1706.88    4504 1703.36  4679.6 1701.63
    4691 1701.99    4770 1700.59  4793.7 1701.12  4834.7  1699.9  4949.9 1698.94
  4977.6 1697.24  4985.5 1696.27  4996.9 1693.28  4999.7 1692.78  5002.9 1693.28
  5014.2 1696.22  5020.7  1697.1  5078.3 1699.21  5148.6  1699.2    5163 1699.69
  5198.2 1699.13  5241.4 1700.62  5291.5 1699.03  5354.9 1701.03  5390.1  1701.3
  5433.3 1703.44  5482.9 1704.72  5532.4 1707.38  5540.4 1708.71  5583.2 1708.87
#Mann= 4 ,-1 , 0
  4227.5      .1       0  4996.9     .07       0  5002.9      .1       0
  5291.5     .05       0
Bank Sta=4996.9,5002.9
XS Rating Curve= 0 ,0
Exp/Cntr=0.3,0.1

Type RM Length L Ch R = 1 ,19173   ,207,207,207
BEGIN DESCRIPTION:
UNT007 IN NNOGR 39.0
END DESCRIPTION:
XS GIS Cut Line= 3
      2774203.09     10069682.06      2773933.97     10069178.54
      2772953.23     10068857.42
#Sta/Elev= 30
  4249.4 1696.25  4442.7 1694.41  4502.9 1692.84  4628.9 1691.25  4694.7 1691.32
  4826.1 1689.73  4979.5 1690.95  4984.8 1690.76  4994.5 1688.69    5002 1688.19
  5004.7 1687.69    5008 1688.19  5011.4 1690.65  5016.7  1690.8  5120.7 1689.56
  5183.9 1689.43  5257.5 1691.16  5278.6 1690.98  5298.1 1692.15  5335.2 1691.85
  5394.6  1692.7  5436.4 1693.95    5489 1694.47    5590 1697.82  5685.5 1699.88
  5722.7 1699.86  5754.5 1700.66  5781.1 1702.03  5818.2 1702.18  5852.3    1704
#Mann= 4 ,-1 , 0
  4249.4      .1       0    5002     .07       0    5008      .1       0
  5394.6     .05       0
Bank Sta=5002,5008
XS Rating Curve= 0 ,0
Exp/Cntr=0.3,0.1

Type RM Length L Ch R = 1 ,18966   ,141,141,141
BEGIN DESCRIPTION:
Mapping XS 3a5122b4
END DESCRIPTION:
XS GIS Cut Line= 3
      2774354.68     10069480.36      2774151.54     10069138.33
      2773056.03     10068692.14
#Sta/Elev= 30
  4115.4 1691.16  4154.6 1690.89  4160.4 1691.48    4176 1690.45  4234.4 1690.25
  4308.5 1688.76  4374.4 1688.24  4394.2 1688.46  4489.7  1687.1  4624.5 1688.23
  4743.3 1687.95  4904.8 1689.93  4910.2  1689.3    4970 1689.56  4987.8 1686.89
  4993.2 1687.41  4999.4 1686.66  5002.2 1686.16  5005.4 1686.66  5011.8 1687.94
  5017.2  1686.7    5024 1688.28  5034.8 1688.85  5056.4  1687.9  5118.8 1690.14
  5124.2 1689.59  5172.4 1690.67  5201.8  1690.6  5218.4 1691.58  5696.1  1700.8
#Mann= 4 ,-1 , 0
  4115.4      .1       0  4374.4     .05       0  4999.4     .04       0
  5005.4     .05       0
Bank Sta=4999.4,5005.4
XS Rating Curve= 0 ,0
Exp/Cntr=0.3,0.1

Type RM Length L Ch R = 1 ,18825   ,326,326,326
BEGIN DESCRIPTION:
Mapping XS a7dea1d5
END DESCRIPTION:
XS GIS Cut Line= 3
      2774369.37     10069429.84      2774288.45     10069100.14
      2773052.99     10068551.71
#Sta/Elev= 30
  3998.1 1690.24  4121.8 1688.42  4241.2  1686.7  4251.5    1686  4275.9 1687.04
  4312.3 1685.52  4411.7 1686.22  4440.6  1685.8  4463.8 1686.54  4539.1 1687.09
  4585.6 1686.82  4637.6 1687.33  4736.2  1686.8    4858 1687.68    4910 1687.17
  4950.3 1687.59  4956.5 1687.49  4972.1 1685.57  4979.7 1683.54  4985.2 1683.25
    4991 1681.98  4993.8 1681.48    4997 1681.98  5031.7 1685.53  5037.8 1687.08
    5191 1689.72  5252.1 1690.11  5379.3 1692.84  5547.7 1695.51  5689.3 1698.76
#Mann= 5 ,-1 , 0
  3998.1      .1       0  4121.8     .05       0  4411.7      .1       0
    4991     .07       0    4997      .1       0
Bank Sta=4991,4997
XS Rating Curve= 0 ,0
Exp/Cntr=0.3,0.1

Type RM Length L Ch R = 1 ,18499   ,466,466,466
BEGIN DESCRIPTION:
UNT007 IN NNOGR 38.0
END DESCRIPTION:
XS GIS Cut Line= 3
      2774484.88     10069171.32      2773873.77     10068553.26
       2773278.1     10068370.62
#Sta/Elev= 30
  4021.4 1685.71  4024.2    1686  4031.3 1685.43  4136.8 1684.27  4162.5 1684.17
    4201 1684.03  4222.2 1683.41  4257.5  1683.7  4328.3 1683.25  4429.4 1683.78
  4568.7 1683.69  4674.8 1682.69  4780.8 1683.45    4917 1683.35  4954.6 1684.16
  4974.4 1683.92  4979.8 1682.31  4990.2 1681.41  5029.1 1681.06  5031.8 1680.56
  5035.1 1681.06  5056.4 1683.64  5072.6 1684.58  5112.5    1685  5199.4 1686.28
  5246.8 1687.72  5312.3 1688.88  5453.2 1690.64  5486.5 1691.32  5513.6 1693.03
#Mann= 10 ,-1 , 0
  4021.4      .1       0  4136.8     .05       0  4162.5     .16       0
  4429.4     .05       0  4954.6     .16       0  5029.1     .07       0
  5035.1     .16       0  5056.4     .05       0  5112.5     .16       0
  5453.2     .05       0
Bank Sta=5029.1,5035.1
XS Rating Curve= 0 ,0
Exp/Cntr=0.3,0.1

Type RM Length L Ch R = 1 ,18033   ,485,485,485
BEGIN DESCRIPTION:
UNT007 IN NNOGR 37.0
END DESCRIPTION:
XS GIS Cut Line= 3
      2774613.34     10068976.85       2774231.4     10068350.14
      2773826.88     10067999.44
#Sta/Elev= 30
  4032.9 1681.31  4147.9 1679.71  4242.8 1679.36  4380.3 1679.76  4481.6 1678.93
  4554.6 1679.46  4728.9 1678.23  4773.2 1679.05  4780.8 1679.76    4795 1678.74
  4855.4 1679.31  4949.4 1680.01  4971.6 1678.49  4993.5 1678.05  4997.1 1677.23
  4999.9 1676.73  5003.1 1677.23  5013.5 1678.57    5022  1679.3  5106.5 1678.96
  5120.8 1679.36    5135 1680.83  5171.5 1680.74  5184.4 1680.46  5241.4 1681.79
  5262.3 1681.45  5276.5 1684.19  5290.8 1688.56  5297.8 1690.05  5302.2 1690.05
#Mann= 7 ,-1 , 0
  4032.9     .05       0  4855.4      .1       0  4997.1     .07       0
  5003.1      .1       0  5013.5     .16       0  5171.5     .05       0
  5290.8      .1       0
Bank Sta=4997.1,5003.1
XS Rating Curve= 0 ,0
Exp/Cntr=0.3,0.1

Type RM Length L Ch R = 1 ,17548   ,416,416,416
BEGIN DESCRIPTION:
UNT007 IN NNOGR 36.0
END DESCRIPTION:
XS GIS Cut Line= 4
      2774654.24     10068628.72      2774611.61     10068339.72
      2774151.54     10067678.26      2773905.06     10067593.21
#Sta/Elev= 30
    4126 1677.49  4150.9 1677.71  4262.5 1676.54  4373.6 1677.04  4393.9 1676.03
  4402.2  1675.9  4407.2 1676.62  4453.7 1675.53  4589.9 1674.45  4713.1 1674.86
  4745.4 1674.41  4795.6 1673.74  4798.3 1673.24  4801.6 1673.74  4824.2 1674.14
  4958.5 1675.39  4998.4 1674.39  5021.6 1674.86  5063.9 1675.87  5093.6 1675.31
  5120.6 1676.18  5161.2 1676.07  5171.2 1676.52  5192.8 1675.87    5248 1677.55
  5279.2 1676.66  5310.4 1678.56  5341.6 1678.98  5372.8 1680.49  5484.6 1682.32
#Mann= 11 ,-1 , 0
    4126     .16       0  4150.9     .05       0  4453.7      .1       0
  4713.1     .16       0  4745.4      .1       0  4795.6     .07       0
  4801.6      .1       0  4824.2     .16       0  4958.5      .1       0
  5021.6     .05       0  5161.2      .1       0
Bank Sta=4795.6,4801.6
XS Rating Curve= 0 ,0
Exp/Cntr=0.3,0.1

Type RM Length L Ch R = 1 ,17132   ,378,378,378
BEGIN DESCRIPTION:
Mapping XS d6df090b
END DESCRIPTION:
XS GIS Cut Line= 4
       2774625.5     10068180.01      2774602.93     10067726.87
      2774573.42     10067627.92      2774214.05     10067416.11
#Sta/Elev= 30
  4382.4 1674.47  4458.8  1674.4  4488.8 1675.48    4619 1674.51  4624.2 1674.29
  4629.2  1672.8    4684 1673.76  4749.1 1674.34  4799.2 1673.06  4824.8 1671.68
  4829.8 1673.56  4842.4 1673.92  4860.2  1673.3  4867.3  1671.6  4872.6 1673.28
  4933.3 1673.82  4938.9  1671.9  4954.2 1670.61  4968.3 1667.77  4975.6 1666.12
  4981.4 1663.64    4999 1661.87  5000.1 1661.74  5002.9 1661.24  5006.1 1661.74
  5012.7 1662.83  5026.4 1668.86  5068.6 1671.23  5188.4 1674.19  5356.5 1677.03
#Mann= 7 ,-1 , 0
  4382.4      .1       0    4684     .16       0  4842.4      .1       0
    4999     .05       0  5000.1    .035       0  5006.1     .05       0
  5068.6      .1       0
Bank Sta=5000.1,5006.1
XS Rating Curve= 0 ,0
Exp/Cntr=0.3,0.1

Type RM Length L Ch R = 1 ,16754   ,271,271,271
BEGIN DESCRIPTION:
UNT007 IN NNOGR 35.0
END DESCRIPTION:
XS GIS Cut Line= 4
      2774760.77      10067856.7      2774795.49     10067533.82
      2774750.35     10067394.93      2774563.12     10067280.52
#Sta/Elev= 30
  4632.1 1669.37  4695.4 1668.16  4735.7 1668.36  4806.1 1666.63  4856.4 1665.96
  4866.4 1665.15  4886.5 1662.07  4896.6  1660.9  4946.9 1656.29  4958.2 1655.87
  4959.5 1655.87  4959.8 1655.37  4962.5 1654.87  4965.8 1655.37  5009.5 1656.08
    5020  1659.3  5026.7 1664.72  5031.9 1664.89  5041.1 1667.35  5063.1 1667.27
  5192.2 1670.27  5207.7 1671.33  5215.8 1671.19    5229 1670.86  5236.3 1671.57
  5280.9 1672.08  5287.1 1672.47  5292.9 1672.26    5316 1672.56  5322.3 1673.16
#Mann= 7 ,-1 , 0
  4632.1      .1       0  4958.2     .16       0  4959.8     .07       0
  4965.8     .16       0  5063.1     .05       0  5215.8      .1       0
  5236.3     .05       0
Bank Sta=4959.8,4965.8
XS Rating Curve= 0 ,0
Exp/Cntr=0.3,0.1

Type RM Length L Ch R = 1 ,16483   ,86,86,86
BEGIN DESCRIPTION:
Mapping XS 240e1ce9
END DESCRIPTION:
XS GIS Cut Line= 4
      2775072.68     10067958.85      2775020.59     10067572.56
      2774948.98     10067375.08      2774658.18      10067264.4
#Sta/Elev= 30
  4524.2 1666.61  4549.5  1665.6  4630.3 1664.63  4731.2 1664.32  4744.6  1665.2
  4761.4 1663.76  4811.9 1662.95  4862.4 1664.48  4895.1  1663.9    4916 1664.43
  4931.8  1656.5  4937.1 1654.49  4946.7 1652.81  4962.4  1651.4  4967.7 1652.44
    4993 1649.77  4998.4 1650.41  5005.5 1649.74  5008.2 1649.24  5011.5 1649.74
    5053 1654.63  5072.3 1656.08  5084.9 1658.24  5104.2 1660.04  5115.5 1664.24
  5122.1 1665.56  5166.5 1666.49  5332.5 1669.33  5396.2 1669.96  5435.2 1671.19
#Mann= 7 ,-1 , 0
  4524.2      .1       0  4946.7     .16       0  5005.5     .07       0
  5011.5     .16       0    5053      .1       0  5166.5     .05       0
  5332.5      .1       0
Bank Sta=5005.5,5011.5
XS Rating Curve= 0 ,0
Exp/Cntr=0.3,0.1

Type RM Length L Ch R = 1 ,16397   ,60,60,60
BEGIN DESCRIPTION:
Mapping XS 1843fe18
END DESCRIPTION:
XS GIS Cut Line= 4
      2775126.93     10067958.88      2775073.27     10067474.79
      2775010.77      10067311.6      2774733.23     10067276.91
#Sta/Elev= 30
  4477.1  1666.2  4572.8  1665.2  4613.1  1664.1  4673.4 1664.19  4689.3 1663.63
  4703.6 1664.19  4723.7 1662.92    4764 1662.44  4821.1 1663.75  4844.5 1663.87
  4875.6 1663.21  4901.9 1661.47  4904.6 1660.97  4907.9 1661.47    4935 1663.07
  4961.3    1667  4986.4 1667.74  4991.8 1666.55  4995.3 1666.79  5016.5 1667.52
  5021.8 1666.64  5046.5 1668.23  5071.2 1666.99  5076.6  1667.7  5101.3 1666.02
  5106.6 1666.42  5131.3 1665.09  5270.4 1667.36  5396.6 1669.32  5418.6 1669.65
#Mann= 7 ,-1 , 0
  4477.1      .1       0  4821.1     .05       0  4901.9     .07       0
  4907.9     .05       0  4995.3      .1       0  5270.4     .05       0
  5396.6      .1       0
Bank Sta=4901.9,4907.9
XS Rating Curve= 0 ,0
Exp/Cntr=0.3,0.1

Type RM Length L Ch R = 1 ,16337   ,319,319,319
BEGIN DESCRIPTION:
UNT007 IN NNOGR 34.0
END DESCRIPTION:
XS GIS Cut Line= 4
      2775166.31     10067794.35      2775119.25     10067431.77
      2775061.72     10067285.33       2774686.9     10067210.36
#Sta/Elev= 30
    4607 1663.71  4668.1  1663.6  4710.2 1661.35  4718.5 1662.07  4808.8 1662.86
  4849.6 1662.57  4863.5  1661.5  4869.8  1658.3  4879.9 1656.96    4890 1660.59
  4910.1 1663.08  4942.6 1661.96  4950.5 1661.09    4956  1658.5  4960.6 1656.33
  4987.5 1650.91  4992.9 1651.59  5008.9 1650.43  5011.7 1649.93  5014.9 1650.43
  5017.3 1652.22    5035 1657.85  5041.7 1661.73  5071.5  1665.1  5088.7 1664.73
  5095.9 1663.58  5110.2 1663.63  5338.3  1667.5  5366.3 1668.25  5512.2 1670.15
#Mann= 7 ,-1 , 0
    4607      .1       0  4808.8     .05       0    4956      .1       0
  5008.9     .07       0  5014.9      .1       0  5338.3     .05       0
  5366.3      .1       0
Bank Sta=5008.9,5014.9
XS Rating Curve= 0 ,0
Exp/Cntr=0.3,0.1

Type RM Length L Ch R = 1 ,16018   ,71,71,71
BEGIN DESCRIPTION:
UNT007 IN NNOGR 33.0
END DESCRIPTION:
XS GIS Cut Line= 4
      2775665.11     10067683.21      2775452.45     10067362.06
       2775194.2     10067255.72      2774777.57     10067197.13
#Sta/Elev= 30
  4543.9 1660.79  4562.1 1660.39  4641.3 1658.99  4692.5 1657.37  4743.6 1656.91
  4779.7 1657.27  4836.9 1658.91  4888.2 1658.57  4938.3 1657.49    4955 1654.13
  4962.3 1651.57  4967.7 1651.05  4983.2 1648.02  4985.9 1647.52  4989.2 1648.02
  4991.6 1648.83  4998.3 1648.19  5015.6 1648.03  5030.7 1649.93  5039.5 1651.54
  5052.4 1656.27  5068.9 1660.41  5074.3 1660.79  5092.8 1661.26  5098.2 1660.72
  5122.2 1660.67  5151.5 1661.59  5385.8 1664.67    5549  1667.6  5629.1 1669.01
#Mann= 6 ,-1 , 0
  4543.9     .05       0  4562.1      .1       0  4888.2     .05       0
  4983.2    .035       0  4989.2     .05       0    5549      .1       0
Bank Sta=4983.2,4989.2
XS Rating Curve= 0 ,0
Exp/Cntr=0.3,0.1

Type RM Length L Ch R = 1 ,15947   ,74,74,74
BEGIN DESCRIPTION:
Mapping XS a4a900fe
END DESCRIPTION:
XS GIS Cut Line= 4
      2775693.34     10067626.81      2775465.63     10067294.24
      2775309.38     10067217.85      2774816.32     10067172.71
#Sta/Elev= 30
  4537.6 1659.92  4608.1 1658.64  4637.9 1658.66  4694.7 1656.86  4727.6 1656.37
  4730.4 1655.87  4733.6 1656.37  4808.4 1658.07  4853.2 1657.56  4875.8 1657.74
    4904 1657.41    4917 1657.83    4931 1659.01  4937.9 1660.36  4953.7 1661.44
  4970.6  1660.4  4976.2 1660.69  4993.2  1660.2  4998.7 1659.41  5004.3 1660.54
  5015.4 1660.31  5021.2 1659.76  5026.8 1660.98  5037.7 1660.82  5071.8 1658.54
  5212.7 1662.35  5336.4 1663.62    5543 1667.38  5567.6 1667.48  5609.7 1668.19
#Mann= 5 ,-1 , 0
  4537.6      .1       0  4727.6    .035       0  4733.6      .1       0
  4875.8     .05       0  5567.6      .1       0
Bank Sta=4727.6,4733.6
XS Rating Curve= 0 ,0
Exp/Cntr=0.3,0.1

Type RM Length L Ch R = 1 ,15873   ,231,231,231
BEGIN DESCRIPTION:
Mapping XS e341e99b
END DESCRIPTION:
XS GIS Cut Line= 4
      2775684.66      10067474.9      2775515.39      10067242.7
       2775339.6     10067142.87      2774814.38     10067112.49
#Sta/Elev= 30
  4628.3 1658.02  4662.5 1657.12  4691.6 1655.22  4748.2 1654.37  4783.8 1655.53
  4798.4 1654.77  4813.1    1655  4854.8 1657.06  4871.6 1656.48  4898.9 1655.81
  4920.8 1657.04  4948.1 1651.93    4964 1651.63  4969.8 1650.48  4979.9 1649.96
  4985.6 1648.68  5001.5 1648.01    5007 1647.02  5023.1 1650.94  5028.9 1651.77
  5044.8 1656.83  5050.5 1657.54    5088 1657.24  5186.8 1661.01  5239.1 1661.62
  5269.2 1660.97  5319.3 1662.49  5506.4  1665.7  5589.8    1667  5643.9 1667.75
#Mann= 6 ,-1 , 0
  4628.3      .1       0  4871.6     .05       0    4964    .035       0
  5023.1     .05       0  5506.4      .1       0  5589.8     .05       0
#XS Ineff= 2 , 0
          4853.2    1657
Permanent Ineff=
       F       F
Bank Sta=4964,5023.1
XS Rating Curve= 0 ,0
Exp/Cntr=0.3,0.1

Type RM Length L Ch R = 1 ,15642   ,215,215,215
BEGIN DESCRIPTION:
UNT007 IN NNOGR 32.0
END DESCRIPTION:
XS GIS Cut Line= 3
        2775792.     10067408.79      2775667.02     10067075.49
       2775296.9     10066867.95
#Sta/Elev= 30
  4569.3  1656.9  4622.4 1656.54  4677.6 1655.41  4702.5  1655.6  4707.9 1655.98
  4713.5 1655.57    4763 1654.81    4788 1654.78  4793.3 1655.23  4818.2 1655.02
  4823.6 1655.41  4878.7 1653.82  4903.7 1653.78    4909 1653.07  4927.3 1652.13
  4946.5 1646.48  4961.6 1645.28  4996.3 1645.19    4999 1644.69  5002.3 1645.19
  5026.8 1645.48  5036.9 1646.27  5049.7 1649.63  5064.3 1652.62  5072.6 1653.75
  5080.3 1654.24  5188.7 1654.97  5272.5 1657.49  5323.3 1658.51  5349.6 1658.55
#Mann= 4 ,-1 , 0
  4569.3      .1       0  4996.3     .07       0  5002.3      .1       0
  5272.5     .05       0
Bank Sta=4996.3,5002.3
XS Rating Curve= 0 ,0
Exp/Cntr=0.3,0.1

Type RM Length L Ch R = 1 ,15427   ,52,52,52
BEGIN DESCRIPTION:
Mapping XS f4dc39a7
END DESCRIPTION:
XS GIS Cut Line= 4
      2775864.78     10067392.45      2775840.63     10067106.74
       2775594.1     10066592.85      2775335.31     10066561.28
#Sta/Elev= 30
  4457.2 1655.68  4471.9 1655.31  4616.5 1654.73  4736.9 1653.18  4847.1 1652.72
  4875.4 1652.19    4881 1652.46  4898.1  1651.5  4913.6 1652.34  4920.8 1653.49
  4926.3 1653.59  4935.8 1652.87  4943.4 1651.01  4948.9 1650.09    4958 1647.65
  4966.1  1646.1  4971.6 1645.37  4977.2 1645.18  4979.9 1644.68  4983.2 1645.18
  4990.3 1645.31  5016.9 1645.34    5034 1646.57  5039.6 1646.22  5056.7 1649.28
  5091.1 1651.21  5175.5  1651.2  5294.3  1653.8  5440.5 1654.15  5574.6 1654.94
#Mann= 4 ,-1 , 0
  4457.2      .1       0  4977.2    .035       0  4983.2      .1       0
  4990.3     .05       0
Bank Sta=4977.2,4983.2
XS Rating Curve= 0 ,0
Exp/Cntr=0.3,0.1

Type RM Length L Ch R = 1 ,15375   ,57,57,57
BEGIN DESCRIPTION:
Mapping XS 2c630df2
END DESCRIPTION:
XS GIS Cut Line= 4
      2775901.67     10067396.82      2775885.77     10067078.96
      2775641.25     10066578.64      2775326.54     10066541.74
#Sta/Elev= 30
  4437.4  1655.7  4598.6 1653.97  4831.5 1652.44    4871 1651.37  4899.1 1652.77
  4906.2 1653.76  4921.6 1654.27  4944.1 1653.85  4961.1 1654.19  4966.6 1653.28
  4983.6 1653.95  4989.1 1652.75  5006.1  1653.4  5011.7 1652.23  5017.5 1652.98
  5028.6 1653.44  5038.5 1653.08  5050.9 1653.03  5062.3 1651.24  5079.2 1649.77
  5098.7 1649.63  5101.5 1649.13  5104.7 1649.63  5107.3 1650.26  5129.8 1650.89
  5184.4 1650.68  5274.8  1652.8    5351 1653.62  5487.5 1653.78  5629.4 1654.85
#Mann= 6 ,-1 , 0
  4437.4      .1       0  5038.5     .05       0  5098.7     .07       0
  5104.7     .05       0  5274.8      .1       0    5351     .05       0
Bank Sta=5098.7,5104.7
XS Rating Curve= 0 ,0
Exp/Cntr=0.3,0.1

Type RM Length L Ch R = 1 ,15318   ,489,489,489
BEGIN DESCRIPTION:
UNT007 IN NNOGR 31.0
END DESCRIPTION:
XS GIS Cut Line= 2
      2776080.29     10067230.15      2775635.61     10066532.04
#Sta/Elev= 30
  4537.5 1653.13  4659.8 1651.88  4782.2 1651.69  4790.2 1652.25  4811.3 1652.17
  4847.7 1650.78  4899.4 1649.85  4935.8 1649.94  4962.8 1651.01  4971.9 1649.78
  4993.3 1645.46  4999.2  1645.8  5011.5  1642.6  5014.2  1642.1  5017.5  1642.6
  5020.4 1644.43  5029.7 1643.71  5035.6 1645.56  5043.1 1645.38  5060.4 1649.43
    5072 1650.64  5087.3 1644.38  5102.4 1643.61  5108.4 1648.01  5123.7 1649.16
  5129.6 1649.02  5137.9 1650.15  5226.1 1651.26  5296.4 1653.18  5365.2 1653.19
#Mann= 5 ,-1 , 0
  4537.5      .1       0  5011.5     .07       0  5017.5      .1       0
  5060.4     .05       0  5226.1      .1       0
Bank Sta=5011.5,5017.5
XS Rating Curve= 0 ,0
Exp/Cntr=0.3,0.1

Type RM Length L Ch R = 1 ,14829   ,594,594,594
BEGIN DESCRIPTION:
Mapping XS f88daa6f
END DESCRIPTION:
XS GIS Cut Line= 4
      2776287.93      10067021.3      2776144.73     10066793.48
      2776092.64     10066637.23      2775669.43     10066489.65
#Sta/Elev= 30
  4826.7 1653.33  4853.6 1651.14  4911.3 1649.21  4926.6 1647.96  4941.9 1645.88
  4963.1    1641    4969 1640.62  4984.3 1636.83  4996.6  1636.4  4999.4  1635.9
  5002.6  1636.4  5005.6  1636.5  5020.9 1641.13  5026.8 1640.99  5036.2  1642.3
  5042.1 1642.22  5048.2 1644.16  5057.4 1643.73  5063.3 1644.37  5078.6 1643.12
  5084.5 1644.15  5106.1 1645.28  5158.3 1646.19  5169.1 1645.82  5211.5 1644.99
  5314.6 1646.96    5339 1646.67  5526.8 1651.12  5597.4 1651.78  5708.7 1652.75
#Mann= 5 ,-1 , 0
  4826.7      .1       0  4996.6     .07       0  5002.6      .1       0
  5169.1     .05       0  5597.4      .1       0
Bank Sta=4996.6,5002.6
XS Rating Curve= 0 ,0
Exp/Cntr=0.3,0.1

Type RM Length L Ch R = 1 ,14235   ,119,119,119
BEGIN DESCRIPTION:
UNT007 IN NNOGR 30.0
END DESCRIPTION:
XS GIS Cut Line= 3
      2776333.53     10066941.01      2776311.83     10066270.48
      2776018.82     10066159.78
#Sta/Elev= 30
  4527.6 1651.31  4644.9 1647.74    4765 1645.83    4785 1644.93    4805 1644.68
  4834.3  1645.4    4855 1644.21  4875.1 1641.41  4885.1 1643.05  4905.1 1642.21
  4935.1 1639.68  4952.3 1637.02  4975.1 1634.52  5002.1 1633.76  5004.9 1633.26
  5008.1 1633.76  5015.1 1636.07  5025.1 1640.74  5035.1 1643.38  5045.1 1643.71
  5055.2 1642.87  5065.2 1643.14  5085.2 1644.83  5285.3 1645.52  5370.5 1646.27
  5375.8 1646.72  5425.5 1647.41  5430.8 1646.65  5474.5 1646.79  5511.7 1647.02
#Mann= 5 ,-1 , 0
  4527.6      .1       0  4952.3     .05       0  5002.1    .035       0
  5008.1     .05       0  5474.5      .1       0
Bank Sta=5002.1,5008.1
XS Rating Curve= 0 ,0
Exp/Cntr=0.3,0.1

Type RM Length L Ch R = 1 ,14116   ,518,518,518
BEGIN DESCRIPTION:
UNT007 IN NNOGR 29.0
END DESCRIPTION:
XS GIS Cut Line= 3
      2776411.65     10066915.02      2776385.61     10066255.29
      2776093.08     10066153.44
#Sta/Elev= 30
  4468.7 1650.82  4630.1 1647.23  4700.2 1645.26  4730.2 1643.86  4810.3 1643.87
  4820.3 1643.62  4840.3 1641.71  4870.3 1641.91  4900.3 1640.31  4932.6 1641.04
  4950.4 1640.05  4960.4 1638.79  4980.4 1633.53  4987.4 1632.83  4990.1 1632.33
  4993.4 1632.83  5020.4 1633.95  5040.4 1636.33  5060.4 1641.66  5070.5 1643.17
  5136.5 1643.01  5145.3 1643.56  5150.6 1643.33  5157.7 1644.42  5189.5  1645.6
  5207.5 1645.03  5263.6 1645.38  5326.6 1646.68  5331.9 1646.19  5438.7 1647.04
#Mann= 3 ,-1 , 0
  4468.7     .05       0  4987.4     .04       0  4993.4     .05       0
Bank Sta=4987.4,4993.4
XS Rating Curve= 0 ,0
Exp/Cntr=0.3,0.1

Type RM Length L Ch R = 1 ,13598   ,695,695,695
BEGIN DESCRIPTION:
UNT007 IN NNOGR 28.0
END DESCRIPTION:
XS GIS Cut Line= 3
      2777024.63     10066203.95      2776573.27     10066006.04
       2776257.4     10066158.77
#Sta/Elev= 30
  4728.6 1646.39    4869 1645.71    4926 1644.84  4962.4 1643.72  4967.9 1642.27
  4985.8 1632.88  4994.4 1629.91  4997.1 1629.41  5000.4 1629.91  5014.7 1632.25
    5038 1634.41  5043.5 1634.32  5061.4    1637  5084.7 1637.23  5113.6 1638.94
  5142.4 1638.38  5165.8 1638.74  5173.4 1641.07  5189.2 1645.93  5194.6 1645.07
  5207.2 1645.86    5230 1645.57    5247 1641.09  5260.1 1639.28    5284 1639.44
  5416.3 1641.62  5455.9 1641.57  5501.1 1643.69  5529.3 1645.81  5572.3 1646.02
#Mann= 7 ,-1 , 0
  4728.6     .05       0    4926      .1       0  4994.4     .07       0
  5000.4      .1       0  5173.4     .05       0  5207.2      .1       0
    5284     .05       0
Bank Sta=4994.4,5000.4
XS Rating Curve= 0 ,0
Exp/Cntr=0.3,0.1

Type RM Length L Ch R = 1 ,12903   ,301,301,301
BEGIN DESCRIPTION:
UNT007 IN NNOGR 27.0
END DESCRIPTION:
XS GIS Cut Line= 3
      2777003.83     10065693.55      2776607.99     10065558.13
      2776223.02      10065800.9
#Sta/Elev= 30
  4434.5 1640.95  4443.9 1640.94  4541.3 1640.81  4572.6 1639.76  4619.8 1639.78
  4697.8 1637.78    4715 1637.97  4851.9 1633.77  4929.1 1633.65  4944.4 1631.55
  4950.3 1632.22  4965.6 1628.78  4971.5 1629.09  4980.8 1627.23    4999 1626.15
  5001.8 1625.65    5005 1626.15  5023.2 1630.63  5029.6 1634.32    5079  1635.1
  5096.2 1633.89  5117.4 1635.15  5132.7 1634.38  5159.8 1634.78  5169.2 1636.95
  5175.1 1637.05  5190.3 1639.65  5218.8 1638.81  5284.5  1641.4    5308 1641.84
#Mann= 4 ,-1 , 0
  4434.5     .05       0  4443.9      .1       0    4999     .07       0
    5005     .05       0
Bank Sta=4999,5005
XS Rating Curve= 0 ,0
Exp/Cntr=0.3,0.1

Type RM Length L Ch R = 1 ,12602   ,764,764,764
BEGIN DESCRIPTION:
UNT007 IN NNOGR 26.0
END DESCRIPTION:
XS GIS Cut Line= 3
      2777014.25     10065592.86      2776601.04     10065349.79
      2776016.94     10065315.71
#Sta/Elev= 30
    4436 1640.25  4520.6 1639.87  4606.4 1638.29  4680.7 1637.65  4732.8 1636.06
  4760.7  1633.7    4788 1632.76  4825.6  1631.1    4928 1630.79    4958 1630.22
  4968.1 1628.94  4988.1 1625.13  4995.1 1624.47  4997.9 1623.97  5001.1 1624.47
  5008.1 1625.61  5018.2 1628.43  5038.2 1635.12  5048.2 1636.79  5058.2 1637.48
  5098.3 1637.95  5128.3 1637.86  5158.4 1636.68  5178.4 1637.69  5288.6 1638.81
  5308.6  1639.6  5388.8  1640.8  5418.8 1641.03  5451.2 1640.16  5500.5 1641.99
#Mann= 5 ,-1 , 0
    4436     .05       0    4788      .1       0  4995.1     .07       0
  5001.1      .1       0  5098.3     .05       0
Bank Sta=4995.1,5001.1
XS Rating Curve= 0 ,0
Exp/Cntr=0.3,0.1

Type RM Length L Ch R = 1 ,11838   ,46,46,46
BEGIN DESCRIPTION:
Mapping XS 68272c3b
END DESCRIPTION:
XS GIS Cut Line= 4
      2777028.14     10065082.45      2776899.65     10064971.32
      2776767.71     10064978.27      2776443.07     10065202.76
#Sta/Elev= 30
    4779 1634.09  4877.1 1631.29  4905.6 1629.92  4926.4 1627.17  4934.1 1625.27
  4946.4 1623.13    4952 1623.13  4968.8 1621.88  4980.1 1621.31  5017.2 1620.82
  5019.9 1620.32  5023.2 1620.82  5050.2 1621.38  5078.1 1624.32    5084 1624.14
  5104.9 1626.51  5113.7 1628.39  5140.9 1629.57  5170.5 1629.89  5250.3 1632.53
  5328.6 1634.44  5343.5 1633.97  5349.6 1634.34  5358.4 1634.12  5364.5 1634.68
  5379.3  1634.2  5400.3 1634.99  5452.3 1634.51  5471.9  1635.3  5475.7 1635.09
#Mann= 5 ,-1 , 0
    4779     .05       0  4968.8      .1       0  5017.2     .07       0
  5023.2      .1       0  5452.3     .05       0
Bank Sta=5017.2,5023.2
XS Rating Curve= 0 ,0
Exp/Cntr=0.3,0.1

Type RM Length L Ch R = 1 ,11792   ,45,45,45
BEGIN DESCRIPTION:
Mapping XS 468cd450
END DESCRIPTION:
XS GIS Cut Line= 4
       2777028.1      10065033.8      2776899.65     10064929.66
      2776771.18     10064933.13      2776505.33     10065138.31
#Sta/Elev= 30
  4797.3 1633.16  4868.2 1631.24    4897 1629.99  4903.4 1630.12  4911.4 1629.49
  4917.8 1630.28  4925.6 1629.53  4932.2 1628.36  4938.6    1630  4946.6 1629.33
    4953 1630.41  4993.7 1629.75  5083.9 1629.06    5090 1628.06  5095.8 1628.06
  5100.6 1627.11  5107.2 1626.55  5118.5 1626.42  5121.2 1625.92  5124.5 1626.42
  5144.1 1627.16  5157.8 1629.02  5235.6 1630.78  5258.3 1631.67  5328.9  1632.8
  5349.7 1633.49  5357.9  1633.1  5378.7 1633.61  5399.5 1633.21    5427 1633.71
#Mann= 4 ,-1 , 0
  4797.3     .05       0  4993.7      .1       0  5118.5     .07       0
  5124.5      .1       0
Bank Sta=5118.5,5124.5
XS Rating Curve= 0 ,0
Exp/Cntr=0.3,0.1

Type RM Length L Ch R = 1 ,11747   ,331,331,331
BEGIN DESCRIPTION:
UNT007 IN NNOGR 25.0
END DESCRIPTION:
XS GIS Cut Line= 4
      2777047.84      10064981.8      2776897.62     10064885.83
      2776722.32     10064898.35      2776547.56     10065079.35
#Sta/Elev= 30
  4800.2 1632.61    4842  1631.7  4914.8 1628.66  4951.1 1629.01  4965.6 1628.46
  4972.3 1623.86  4975.8 1619.81  4980.5 1619.81  4987.6 1616.36  4994.7 1614.92
  4997.4 1614.42  5000.7 1614.92  5007.7 1615.75    5016 1621.85  5018.7 1621.41
    5021 1621.03  5027.7 1625.12  5057.8 1627.69  5067.8 1626.24  5087.9 1625.23
  5097.9 1622.98  5107.9 1619.69    5118 1619.29    5128 1620.01    5138  1624.4
  5153.6 1624.77  5160.8 1625.64  5167.8 1625.41  5203.3 1628.76  5405.8 1632.75
#Mann= 4 ,-1 , 0
  4800.2     .05       0  4994.7    .035       0  5000.7     .05       0
  5018.7      .1       0
Bank Sta=4994.7,5000.7
XS Rating Curve= 0 ,0
Exp/Cntr=0.3,0.1

Type RM Length L Ch R = 1 ,11416   ,459,459,459
BEGIN DESCRIPTION:
UNT007 IN NNOGR 24.0
END DESCRIPTION:
XS GIS Cut Line= 3
       2777121.9     10064846.36      2776965.63     10064596.32
      2776212.83     10064180.03
#Sta/Elev= 30
  4639.2 1630.22  4668.3 1629.85  4803.8 1625.31  4932.6 1623.96  4948.9 1624.36
  4970.6 1623.26  4986.7 1615.57  4999.4  1612.9  5005.4 1612.73  5008.2 1612.23
  5011.4 1612.73  5022.2 1617.79  5030.2 1622.63  5045.1    1627  5051.9 1627.39
  5057.6 1629.06  5073.7 1629.33  5079.4  1631.4  5089.7 1631.66    5139 1635.87
  5182.5 1637.27  5353.6 1639.31  5404.7  1639.6  5464.3 1638.05  5539.9  1641.2
  5582.2 1641.91  5610.9  1639.9  5626.9 1641.68  5648.7 1642.77  5794.3 1646.08
#Mann= 5 ,-1 , 0
  4639.2     .05       0  4668.3      .1       0  5005.4     .07       0
  5011.4      .1       0  5539.9     .05       0
Bank Sta=5005.4,5011.4
XS Rating Curve= 0 ,0
Exp/Cntr=0.3,0.1

Type RM Length L Ch R = 1 ,10957   ,404,404,404
BEGIN DESCRIPTION:
UNT007 IN NNOGR 23.0
END DESCRIPTION:
XS GIS Cut Line= 2
      2777354.52     10064787.33       2777212.5     10064167.28
#Sta/Elev= 30
  4697.7 1630.22  4704.5 1630.34  4742.3 1628.58  4747.4 1628.89  4773.2 1627.79
  4795.4 1627.36  4870.2 1625.11  4929.3 1624.06  4967.1 1620.97  4972.2 1619.91
  4978.4 1616.11  4988.6 1610.57  4995.9 1609.04  4998.6 1608.54  5001.9 1609.04
  5009.2 1609.62  5015.1 1612.13  5020.3 1612.36  5029.7 1615.94  5039.9 1618.45
    5058 1621.95  5063.2 1622.77  5070.7 1623.48  5100.9 1625.15  5111.7 1626.08
  5204.1 1630.98  5234.8 1631.94  5275.9 1633.67  5325.8 1634.86  5333.8 1635.27
#Mann= 4 ,-1 , 0
  4697.7     .05       0  4870.2      .1       0  4995.9     .07       0
  5001.9      .1       0
Bank Sta=4995.9,5001.9
XS Rating Curve= 0 ,0
Exp/Cntr=0.3,0.1

Type RM Length L Ch R = 1 ,10553   ,449,449,449
BEGIN DESCRIPTION:
UNT007 IN NNOGR 22.0
END DESCRIPTION:
XS GIS Cut Line= 3
      2777670.49     10064870.67      2777684.38      10064311.6
      2777580.62     10064017.62
#Sta/Elev= 30
  4573.1 1630.83  4640.1  1629.6  4689.1 1627.46  4694.1  1627.8  4780.1 1624.69
  4862.1 1621.29  4870.1  1621.1  4880.1 1621.56  4920.1  1618.9  4930.2 1619.11
  4940.2 1617.73  4950.2  1614.4  4980.2 1606.63  4997.2 1603.89  4999.9 1603.39
  5003.2 1603.89  5010.2 1607.39  5020.2 1614.18  5030.2 1617.26  5040.2 1617.95
  5072.3 1618.76  5095.5  1619.5  5100.5 1619.16  5110.2 1619.86  5132.3 1620.27
  5209.5 1624.81    5228 1625.65    5321 1631.66  5372.1 1633.51  5444.1 1635.08
#Mann= 6 ,-1 , 0
  4573.1     .05       0  4862.1      .1       0  4997.2     .07       0
  5003.2      .1       0  5072.3     .16       0  5209.5      .1       0
Bank Sta=4997.2,5003.2
XS Rating Curve= 0 ,0
Exp/Cntr=0.3,0.1

Type RM Length L Ch R = 1 ,10104   ,348,348,348
BEGIN DESCRIPTION:
UNT007 IN NNOGR 21.0
END DESCRIPTION:
XS GIS Cut Line= 3
      2778219.11     10064634.54      2777986.46     10064113.68
      2777810.73     10063917.27
#Sta/Elev= 30
  4514.4 1627.47  4537.2 1627.73  4567.8 1626.82  4591.9 1626.51  4668.6  1623.9
  4726.6 1621.91  4764.5 1620.09  4831.8 1617.61  4842.7 1617.13  4854.8 1617.17
  4871.4 1616.17  4931.5 1614.79    4941 1614.01  4946.5 1614.18  4953.4 1612.94
  4969.7 1608.86  4975.3 1605.45  4995.4 1602.17  4998.1 1601.67  5001.4 1602.17
  5008.1 1604.26  5021.6 1612.11    5030 1615.12  5039.3 1617.66  5051.9 1619.33
  5062.5 1619.85  5082.1 1621.61  5239.2 1629.39  5288.5 1631.19  5348.4 1632.19
#Mann= 6 ,-1 , 0
  4514.4     .05       0  4567.8      .1       0  4764.5     .16       0
  4831.8      .1       0  4995.4     .07       0  5001.4      .1       0
Bank Sta=4995.4,5001.4
XS Rating Curve= 0 ,0
Exp/Cntr=0.3,0.1

Type RM Length L Ch R = 1 ,9756    ,490,490,490
BEGIN DESCRIPTION:
UNT007 IN NNOGR 20.0
END DESCRIPTION:
XS GIS Cut Line= 3
      2778607.96     10064391.43      2778153.13     10063884.52
      2777901.54     10063832.82
#Sta/Elev= 30
  4624.1 1622.49  4735.4 1620.94  4876.7 1620.28  4890.9 1619.69  4933.5 1616.05
  4947.7 1613.98  4955.2 1611.21  4961.9 1610.97  4969.4 1605.69  4976.1 1605.63
  4983.6 1601.08  4994.2 1598.14  4996.9 1597.64  5000.2 1598.14  5011.3 1602.99
  5018.7    1609  5025.5 1608.22    5033 1611.46  5047.2 1612.05  5053.9 1610.93
  5061.4 1611.72  5068.1 1611.11  5082.3 1613.18    5104 1613.32  5188.4 1616.93
  5210.1 1617.22    5231 1618.62  5273.7  1619.8  5493.7 1628.63    5562 1630.11
#Mann= 3 ,-1 , 0
  4624.1      .1       0  4994.2     .07       0  5000.2      .1       0
Bank Sta=4994.2,5000.2
XS Rating Curve= 0 ,0
Exp/Cntr=0.3,0.1

Type RM Length L Ch R = 1 ,9266    ,421,421,421
BEGIN DESCRIPTION:
UNT007 IN NNOGR 19.0
END DESCRIPTION:
XS GIS Cut Line= 3
      2778791.99     10063738.68      2778507.29     10063676.18
      2778042.77     10063780.18
#Sta/Elev= 30
  4644.4 1618.41  4687.3 1618.46  4736.2 1617.15  4741.4 1616.39  4760.6 1615.82
  4791.3  1613.7  4822.1 1612.74  4852.8    1611  4872.7 1610.63  4883.5 1609.69
  4914.2 1608.91  4921.7 1608.21  4926.5 1608.47  4935.9 1607.99  4948.8 1606.07
  4992.2 1595.93  4994.3 1595.85  4997.1 1595.35  5000.3 1595.85  5016.7  1596.9
  5026.9 1600.06  5035.6 1604.51  5040.7  1605.9  5047.4 1609.02  5067.9 1611.21
  5088.1  1612.5  5127.4 1615.67    5176 1618.59  5267.8 1622.03  5411.9 1626.44
#Mann= 5 ,-1 , 0
  4644.4      .1       0  4926.5     .05       0  4994.3    .035       0
  5000.3     .05       0  5088.1      .1       0
Bank Sta=4994.3,5000.3
XS Rating Curve= 0 ,0
Exp/Cntr=0.3,0.1

Type RM Length L Ch R = 1 ,8845    ,392,392,392
BEGIN DESCRIPTION:
UNT007 IN NNOGR 18.0
END DESCRIPTION:
XS GIS Cut Line= 3
      2779007.28     10063700.48      2778628.82     10063370.63
      2778146.15     10063356.74
#Sta/Elev= 30
  4597.8 1617.02  4793.4 1617.01  4821.7 1616.27  4842.8 1614.42  4934.9 1608.85
  4949.1 1607.36  4963.4 1603.33    4970 1600.39  4984.3  1595.6  4991.9  1594.8
  4995.5 1593.69  4998.2 1593.19  5001.5 1593.69  5012.7 1593.99  5020.3 1595.74
    5027    1598    5034 1602.36  5041.2  1604.9  5047.9 1605.81  5076.3 1606.77
  5102.5 1606.44  5165.5 1610.04  5190.2 1610.49  5220.2 1612.15  5250.2 1612.62
  5270.3 1613.79  5280.3 1613.62  5490.3 1621.82  5509.4 1621.72  5582.7 1623.44
#Mann= 3 ,-1 , 0
  4597.8      .1       0  4995.5     .07       0  5001.5      .1       0
Bank Sta=4995.5,5001.5
XS Rating Curve= 0 ,0
Exp/Cntr=0.3,0.1

Type RM Length L Ch R = 1 ,8453    ,730,730,730
BEGIN DESCRIPTION:
UNT007 IN NNOGR 17.0
END DESCRIPTION:
XS GIS Cut Line= 3
       2779121.9     10063051.18      2778607.99     10063106.74
      2778173.96     10063256.05
#Sta/Elev= 30
  4604.9 1612.76  4708.9 1613.16  4849.8    1605    4881 1603.97  4910.1  1603.2
  4949.8 1600.93  4980.5 1591.54  4997.6 1589.14  5000.4 1588.64  5003.6 1589.14
  5010.7 1590.43  5020.7 1593.78  5026.5 1597.37  5030.8 1600.04  5040.9 1604.54
  5046.6 1605.86  5051.6 1605.56    5071 1607.43  5127.3 1610.54  5142.5 1610.22
  5158.5 1611.34  5163.8 1610.94  5195.5 1612.23  5215.7 1613.58    5221  1613.2
  5283.4 1615.12  5403.1 1619.55  5408.4 1619.06    5528 1621.85  5580.8 1621.57
#Mann= 6 ,-1 , 0
  4604.9     .16       0    4881      .1       0  4997.6     .07       0
  5003.6      .1       0  5026.5     .16       0  5195.5      .1       0
Bank Sta=4997.6,5003.6
XS Rating Curve= 0 ,0
Exp/Cntr=0.3,0.1

Type RM Length L Ch R = 1 ,7723    ,402,402,402
BEGIN DESCRIPTION:
UNT007 IN NNOGR 16.0
END DESCRIPTION:
XS GIS Cut Line= 3
       2779021.2     10062572.02       2778430.9     10062530.35
      2777838.66     10062769.32
#Sta/Elev= 30
  4668.4 1604.28  4786.4 1602.33  4851.6  1600.2  4901.7 1596.24  4911.7 1596.81
  4961.9 1587.42  4971.9 1586.35  4991.9 1585.99    5000 1584.74  5002.8 1584.24
    5006 1584.74    5012 1587.79    5022 1595.02  5031.9 1600.41  5052.1 1603.79
  5192.4 1613.64  5258.9 1617.09  5304.9 1618.17  5310.3 1617.56  5379.5 1620.22
  5441.8 1621.59  5532.4  1622.1  5554.6 1622.77  5573.3  1624.4  5597.1 1622.29
  5704.8 1622.91    5748 1621.27  5780.4 1623.93  5843.4 1624.29  5898.8 1624.87
#Mann= 7 ,-1 , 0
  4668.4     .16       0  4786.4      .1       0    5000     .07       0
    5006      .1       0  5031.9     .16       0  5379.5      .1       0
  5843.4     .05       0
Bank Sta=5000,5006
XS Rating Curve= 0 ,0
Exp/Cntr=0.3,0.1

Type RM Length L Ch R = 1 ,7321    ,521,521,521
BEGIN DESCRIPTION:
UNT007 IN NNOGR 15.0
END DESCRIPTION:
XS GIS Cut Line= 2
      2779177.39     10062405.32      2778649.77     10062068.62
#Sta/Elev= 30
  4769.9 1606.78  4784.3 1606.48  4799.5 1605.15  4820.7 1604.61  4835.9 1603.43
  4841.8 1603.57    4894 1599.18  4914.6 1598.84  4922.8  1597.3  4929.8 1594.54
  4935.8  1593.4    4951 1588.66  4958.4 1587.03    4991 1582.84  4993.8 1582.34
    4997 1582.84  5008.5 1583.64  5023.7 1586.29    5039 1586.71  5053.3 1588.83
  5066.1 1592.54  5075.4 1593.88  5169.3 1601.01  5205.7 1603.15    5248 1604.52
  5263.2 1605.69  5284.4 1605.42  5320.7 1607.16    5375 1608.04  5395.8 1608.59
#Mann= 5 ,-1 , 0
  4769.9     .16       0    4894      .1       0    4991     .07       0
    4997      .1       0    5375     .16       0
Bank Sta=4991,4997
XS Rating Curve= 0 ,0
Exp/Cntr=0.3,0.1

Type RM Length L Ch R = 1 ,6800    ,596,596,596
BEGIN DESCRIPTION:
UNT007 IN NNOGR 14.0
END DESCRIPTION:
XS GIS Cut Line= 3
      2779406.63     10061912.31      2778896.18     10061762.99
       2778368.4     10061985.21
#Sta/Elev= 30
  4688.2 1607.48  4707.1 1607.27  4734.9  1604.7  4740.1 1604.84  4780.1 1601.52
  4827.7 1598.89    4879 1594.96  4894.7  1593.1  4936.3 1589.43  4945.9 1586.44
  4951.1 1586.44  4957.2 1584.51    4978 1581.78  4984.6 1578.67  4989.8 1578.46
  4995.9 1576.66  4998.6 1576.16  5001.9 1576.66  5009.3 1577.64    5018 1580.07
  5023.2 1582.13  5030.1 1588.87  5040.5 1591.82  5134.3 1597.71  5162.2 1598.91
  5287.2 1603.33  5354.7  1604.6  5407.4 1605.43  5699.5 1612.25  5792.7 1612.58
#Mann= 6 ,-1 , 0
  4688.2      .1       0  4827.7     .05       0  4995.9    .035       0
  5001.9     .05       0  5354.7      .1       0  5407.4     .05       0
Bank Sta=4995.9,5001.9
XS Rating Curve= 0 ,0
Exp/Cntr=0.3,0.1

Type RM Length L Ch R = 1 ,6204    ,211,211,211
BEGIN DESCRIPTION:
UNT007 IN NNOGR 13.0
END DESCRIPTION:
XS GIS Cut Line= 2
      2779514.27     10061315.08      2778372.66     10061145.05
#Sta/Elev= 30
  4640.1 1604.38  4666.2  1604.4  4700.4 1602.67  4751.6 1599.01  4777.4  1596.6
  4820.9 1593.85  4890.2 1588.05  4929.1 1586.21  4939.2  1585.1  4949.3 1583.25
  4954.5 1581.13  4959.6 1580.71  4989.7 1575.81  4996.8  1575.3  4999.6  1574.8
  5002.8  1575.3  5009.9 1577.24  5018.8 1583.17  5023.8 1584.09  5030.2 1587.82
  5093.2 1589.88    5291 1601.32  5296.1 1601.23  5429.7 1608.53  5464.9 1609.76
  5505.3 1612.24  5563.3 1614.72  5667.1 1617.68  5790.8 1617.88  5794.3  1617.9
#Mann= 5 ,-1 , 0
  4640.1     .16       0  4700.4      .1       0  4996.8    .035       0
  5002.8      .1       0  5790.8      .1       0
Bank Sta=4996.8,5002.8
XS Rating Curve= 0 ,0
Exp/Cntr=0.3,0.1

Type RM Length L Ch R = 1 ,5993    ,517,517,517
BEGIN DESCRIPTION:
UNT007 IN NNOGR 12.0
END DESCRIPTION:
XS GIS Cut Line= 2
      2779427.43     10061092.85      2778875.37     10061002.58
#Sta/Elev= 30
  4764.2 1598.14  4805.2 1595.96  4844.2 1594.14  4850.5 1593.38  4855.6 1593.46
  4884.7 1591.61  4935.4 1586.77  4945.5 1584.95  4955.7 1581.73  4965.8 1579.22
  4973.2 1576.68  4977.3 1576.26  4993.2 1572.36    4996 1571.86  4999.2 1572.36
  5006.3 1572.72  5016.5 1574.77  5034.6 1579.76  5039.7 1580.41  5046.9 1582.45
  5087.4 1585.32  5101.1  1586.9  5127.9 1588.64  5157.4  1589.8  5162.5 1589.56
  5218.8 1592.19  5223.8 1592.02  5269.8 1594.81  5285.2 1596.22  5323.6 1597.92
#Mann= 5 ,-1 , 0
  4764.2     .05       0  4805.2      .1       0  4977.3     .05       0
  4993.2    .035       0  4999.2     .05       0
Bank Sta=4993.2,4999.2
XS Rating Curve= 0 ,0
Exp/Cntr=0.3,0.1

Type RM Length L Ch R = 1 ,5476    ,437,437,437
BEGIN DESCRIPTION:
UNT007 IN NNOGR 11.0
END DESCRIPTION:
XS GIS Cut Line= 3
      2779541.99     10060662.28      2779212.15     10060544.24
      2778903.26     10060561.59
#Sta/Elev= 30
  4605.6 1592.52  4640.9 1591.44  4737.9 1587.36  4832.4  1584.4  4850.9 1584.48
  4874.9 1583.91  4906.7 1582.52    4928 1579.99  4937.9 1577.38  4943.2 1576.54
  4949.2 1574.73  4969.6 1574.47  4979.6 1573.81  4989.7 1571.42  4996.7 1568.69
  4999.4 1568.19  5002.7 1568.69  5009.7 1568.82  5019.7 1573.66  5029.7 1579.42
  5035.4 1582.17  5040.4 1581.92  5089.8 1586.37  5149.9 1590.62  5159.9 1591.82
  5209.7 1595.79  5214.7 1595.47    5220 1596.38  5250.1 1598.23  5265.3 1599.77
#Mann= 4 ,-1 , 0
  4605.6      .1       0  4737.9     .16       0  4996.7     .07       0
  5002.7     .16       0
Bank Sta=4996.7,5002.7
XS Rating Curve= 0 ,0
Exp/Cntr=0.3,0.1

Type RM Length L Ch R = 1 ,5039    ,496,496,496
BEGIN DESCRIPTION:
UNT007 IN NNOGR 10.0
END DESCRIPTION:
XS GIS Cut Line= 3
      2779646.17     10060457.43      2779396.18     10060197.02
      2779083.72     10060245.62
#Sta/Elev= 30
  4705.4 1589.76  4911.5 1578.75  4968.1 1574.57    4975 1573.03  4982.2 1567.74
  4985.4 1566.93  4993.4 1565.11  4996.2 1564.61  4999.4 1565.11  5003.3 1565.22
  5024.7 1570.69  5031.6 1571.44  5045.8 1574.98    5053 1577.74  5059.9 1578.88
  5073.3 1579.76  5094.4 1579.05  5114.7  1581.6  5124.8 1580.85  5134.9 1581.16
  5141.3 1582.28  5146.3 1581.31  5155.2 1582.36  5175.4 1582.43  5247.4 1587.37
  5286.7 1590.02  5296.8 1589.79    5327 1592.38  5347.4 1592.56  5382.6 1594.31
#Mann= 6 ,-1 , 0
  4705.4      .1       0  4985.4     .05       0  4993.4    .035       0
  4999.4     .05       0  5247.4      .1       0    5327     .05       0
Bank Sta=4993.4,4999.4
XS Rating Curve= 0 ,0
Exp/Cntr=0.3,0.1

Type RM Length L Ch R = 1 ,4543    ,494,494,494
BEGIN DESCRIPTION:
UNT007 IN NNOGR 9.0
END DESCRIPTION:
XS GIS Cut Line= 3
      2779993.37     10059919.23      2779705.21     10059842.85
       2779208.7      10059874.1
#Sta/Elev= 30
  4652.1 1588.74  4693.2 1587.81  4733.4 1586.39  4760.6 1584.63  4773.6  1584.7
    4802 1583.74  4813.8 1582.57  4843.4 1581.09  4848.9 1580.09  4874.4 1579.84
  4915.8 1577.53  4939.8 1576.74  4950.2 1576.18    4957 1573.59    4987 1564.33
    4997 1562.45  5004.1 1562.44  5006.8 1561.94  5010.1 1562.44  5017.1 1564.53
  5039.1 1568.89    5043 1569.95    5048 1570.04  5067.2 1572.54  5097.2 1574.88
  5207.8 1580.76  5257.6 1582.49  5357.5 1588.22  5362.5 1587.94  5447.7 1592.46
#Mann= 5 ,-1 , 0
  4652.1     .05       0  4939.8      .1       0  5004.1     .07       0
  5010.1      .1       0  5039.1     .05       0
Bank Sta=5004.1,5010.1
XS Rating Curve= 0 ,0
Exp/Cntr=0.3,0.1

Type RM Length L Ch R = 1 ,4049    ,266,266,266
BEGIN DESCRIPTION:
UNT007 IN NNOGR 8.0
END DESCRIPTION:
XS GIS Cut Line= 3
      2780097.58     10059756.05      2779864.93     10059415.77
      2779465.62     10059325.49
#Sta/Elev= 30
    4488 1584.94    4511 1584.14    4532  1584.8  4546.9 1583.07  4567.9 1582.75
  4597.7  1580.8  4639.6 1579.76  4684.4 1577.35  4696.7 1577.87    4933 1571.27
  4958.1 1570.91  4968.4 1568.79  4975.5 1565.24  4980.6 1564.32  4988.9 1560.51
  4996.1 1559.25  4998.9 1558.75  5002.1 1559.25  5023.8 1564.66  5033.2 1565.46
  5036.7 1565.56  5040.1 1565.65    5067 1571.83  5072.1 1571.19  5133.4 1574.69
  5163.6 1576.44  5201.6 1579.95  5206.7 1581.39  5233.6 1583.43  5309.6 1589.71
#Mann= 8 ,-1 , 0
    4488     .05       0    4933      .1       0  4996.1     .07       0
  5002.1      .1       0  5033.2     .05       0  5036.7      .1       0
  5133.4     .05       0  5233.6      .1       0
Bank Sta=4996.1,5002.1
XS Rating Curve= 0 ,0
Exp/Cntr=0.3,0.1
