--- UNT007 IN SNOGR.prj (project) ---

Proj Title=UNT007 IN SNOGR Base Level Engineering
Current Plan=p01
Default Exp/Contr=0.3,0.1
English Units
Geom File=g01
Flow File=f01
Plan File=p01
BEGIN DESCRIPTION:
UNT007 IN SNOGR
END DESCRIPTION:

--- UNT007 IN SNOGR.p01 (plan) ---

Plan Title=Multiple Run
Short Identifier=Multiple
Geom File=g01
Flow File=f01
Subcritical Flow
K Sum by GR= 0
Std Step Tol= 0.01
Critical Tol= 0.01
Num of Std Step Trials= 20
Max Error Tol= 0.3
Flow Tol Ratio= 0.001
Split Flow NTrial= 30
Split Flow Tol= 0.02
Split Flow Ratio= 0.02
Log Output Level= 0
Friction Slope Method= 1
Unsteady Friction Slope Method= 2
Unsteady Bridges Friction Slope Method= 1
Parabolic Critical Depth
Global Vel Dist=  1 , 1 , 1
Global Log Level= 0
CheckData=True
Encroach Param= -1, 0, 0, 0
BEGIN DESCRIPTION:
Multiple Run
END DESCRIPTION:

--- UNT007 IN SNOGR.f01 (steady flow) ---

Flow Title=Multiple
Number of Profiles=7
Profile Names=10-year,25-year,50-year,1pct_min,100-year,1pct_plu,500-year
River Rch & RM= UNT007 IN SNOGR,Reach-1,20107
     957    1396    1780    1662    2247    3039    3595
River Rch & RM= UNT007 IN SNOGR,Reach-1,19566
    1337    1968    2522    2362    3194    4319    5144
River Rch & RM= UNT007 IN SNOGR,Reach-1,9259
    1615    2387    3068    2878    3893    5264    6293
Boundary for River Rch & Prof#=UNT007 IN SNOGR,Reach-1,1
Up Type=0
Dn Type=3
Dn Slope=0.005
Boundary for River Rch & Prof#=UNT007 IN SNOGR,Reach-1,2
Up Type=0
Dn Type=3
Dn Slope=0.005
Boundary for River Rch & Prof#=UNT007 IN SNOGR,Reach-1,3
Up Type=0
Dn Type=3
Dn Slope=0.005
Boundary for River Rch & Prof#=UNT007 IN SNOGR,Reach-1,4
Up Type=0
Dn Type=3
Dn Slope=0.005
Boundary for River Rch & Prof#=UNT007 IN SNOGR,Reach-1,5
Up Type=0
Dn Type=3
Dn Slope=0.005
Boundary for River Rch & Prof#=UNT007 IN SNOGR,Reach-1,6
Up Type=0
Dn Type=3
Dn Slope=0.005
Boundary for River Rch & Prof#=UNT007 IN SNOGR,Reach-1,7
Up Type=0
Dn Type=3
Dn Slope=0.005

--- UNT007 IN SNOGR.g01 (geometry) ---

Geom Title=Existing Conditions

River Reach=UNT007 IN SNOGR,Reach-1
Reach XY= 30
      2829748.47     10041493.73      2829403.25     10041880.58
      2829555.73     10042732.43      2829142.14     10043289.95
      2829667.91     10043686.28      2829399.98     10044760.66
      2829676.84     10045138.22      2829369.71     10045513.49
      2829783.35     10045662.06      2829824.39     10045953.08
      2829510.17     10046239.63      2829676.42     10046542.85
      2829309.37     10046744.31      2829558.55     10047138.33
      2828921.96     10047557.77      2829425.10     10048325.15
      2829430.80     10048792.90      2830045.67     10049399.45
      2829554.98     10050695.29      2830325.58     10050699.86
      2830269.57     10051723.28      2830623.61     10052316.60
      2830918.60     10052552.86      2831651.89     10052140.87
      2831481.34     10052588.83      2832042.69     10052814.93
      2832340.75     10053319.10      2832343.56     10053666.41
      2831881.01     10053984.95      2831958.51     10054474.32

Type RM Length L Ch R = 1,20107,541,541,541
BEGIN DESCRIPTION:
UNT007 IN SNOGR 34.0
END DESCRIPTION:
XS GIS Cut Line= 2
      2828631.51     10041536.87      2830329.41     10041562.91
#Sta/Elev= 30
  3901.4 1553.66  3958.4 1550.99  4128.4 1545.97  4428.4 1540.63  4588.4 1536.83
  4658.4 1536.28  4718.5 1533.63  4738.5 1534.47  4818.5 1535.57  4838.5 1535.01
  4858.5 1535.24  4878.5 1534.01  4898.5 1533.83  4928.5 1533.73  4948.5 1534.42
  4978.5 1532.68  4995.5 1530.43  4998.2 1529.93  5001.5 1530.43  5008.5 1530.75
  5028.5 1534.90  5068.5 1540.47  5198.5 1546.91  5228.5 1547.81  5325.4 1553.47
  5388.5 1556.05  5468.5 1560.79  5518.5 1562.96  5548.5 1565.02  5599.5 1567.19
#Mann=3,-1,0
  3901.4    0.05       0  4995.5    0.04       0  5001.5    0.05       0
Bank Sta=4995.5,5001.5
Exp/Cntr=0.3,0.1

Type RM Length L Ch R = 1,19566,152,152,152
BEGIN DESCRIPTION:
UNT007 IN SNOGR 33.0
END DESCRIPTION:
XS GIS Cut Line= 3
      2828406.00     10041690.18      2829243.71     10041885.51
      2830228.95     10041924.57
#Sta/Elev= 30
  3980.8 1559.54  4024.4 1556.69  4055.2 1556.38  4121.3 1553.02  4130.9 1552.68
  4219.5 1549.19  4291.4 1546.40  4311.9 1546.86  4454.7 1542.27  4682.9 1538.18
  4712.4 1538.76  4732.9 1536.95  4805.9 1535.73  4875.8 1533.48  4926.6 1529.44
  4942.8 1529.38  4945.6 1528.88  4948.8 1529.38  4975.8 1530.76  4985.9 1530.77
  4995.9 1529.38  5025.9 1530.64  5177.9 1532.80  5476.5 1546.05  5546.3 1550.34
  5626.4 1553.86  5636.4 1555.22  5666.4 1555.48  5796.5 1561.04  5827.0 1564.78
#Mann=8,-1,0
  3980.8    0.05       0  4121.3     0.1       0  4130.9    0.05       0
  4219.5     0.1       0  4805.9    0.16       0  4942.8    0.07       0
  4948.8    0.16       0  5476.5     0.1       0
Bank Sta=4942.8,4948.8
Exp/Cntr=0.3,0.1

Type RM Length L Ch R = 1,19414,101,101,101
BEGIN DESCRIPTION:
Mapping XS 0052ca26
END DESCRIPTION:
XS GIS Cut Line= 3
      2828313.78     10041885.83      2829256.47     10042062.91
      2830119.55     10041948.52
#Sta/Elev= 30
  3894.8 1556.68  3963.5 1554.33  4001.3 1554.73  4017.7 1553.43  4082.7 1551.17
  4127.9 1550.90  4174.3 1548.83  4245.5 1547.24  4479.5 1539.41  4643.1 1536.97
  4693.2 1536.95  4731.2 1535.27  4815.0 1533.92  4888.5 1533.21  4906.4 1531.23
  4936.7 1525.51  4974.0 1524.32  4976.8 1523.82  4980.0 1524.32  5138.4 1525.00
  5158.6 1526.49  5178.8 1529.26  5187.0 1530.87  5192.1 1533.03  5199.0 1533.57
  5229.2 1533.89  5470.8 1545.59  5495.6 1546.31  5592.4 1552.51  5724.6 1557.58
#Mann=8,-1,0
  3894.8    0.05       0  3963.5     0.1       0  4643.1    0.05       0
  4731.2     0.1       0  4815.0    0.16       0  4974.0    0.07       0
  4980.0    0.16       0  5470.8     0.1       0
Bank Sta=4974,4980
Exp/Cntr=0.3,0.1

Type RM Length L Ch R = 1,19313,126,126,126
BEGIN DESCRIPTION:
Mapping XS 7ba04b2a
END DESCRIPTION:
XS GIS Cut Line= 3
      2828267.09     10041963.62      2829300.13     10042154.60
      2830120.41     10042067.80
#Sta/Elev= 30
  3853.2 1554.57  3927.8 1553.58  4200.4 1547.53  4360.0 1542.04  4547.0 1537.91
  4630.3 1536.42  4674.6 1536.10  4763.1 1533.15  4824.6 1532.93  4848.2 1532.30
  4851.0 1531.80  4854.2 1532.30  4881.7 1533.38  4912.1 1536.23  4942.3 1536.03
  4958.5 1534.17  4963.5 1537.61  4982.5 1536.55  5032.8 1537.92  5051.2 1535.96
  5056.2 1539.08  5149.0 1534.02  5154.0 1536.76  5193.7 1534.03  5233.9 1533.03
  5246.8 1534.64  5274.1 1533.93  5504.0 1545.78  5656.3 1554.18  5728.6 1557.01
#Mann=10,-1,0
  3853.2    0.05       0  3927.8     0.1       0  4360.0    0.05       0
  4547.0     0.1       0  4630.3    0.05       0  4674.6     0.1       0
  4824.6    0.16       0  4848.2    0.07       0  4854.2    0.16       0
  5504.0     0.1       0
Bank Sta=4848.2,4854.2
Exp/Cntr=0.3,0.1

Type RM Length L Ch R = 1,19187,505,505,505
BEGIN DESCRIPTION:
UNT007 IN SNOGR 32.0
END DESCRIPTION:
XS GIS Cut Line= 3
      2828225.20     10042073.32      2829329.39     10042276.45
      2830094.28     10042135.96
#Sta/Elev= 30
  3761.7 1554.98  3785.4 1555.17  3901.1 1550.87  3937.9 1549.99  3998.9 1546.84
  4122.6 1545.58  4253.6 1542.52  4402.9 1539.22  4571.4 1535.96  4622.4 1535.55
  4639.5 1533.99  4770.5 1532.12  4822.5 1531.67  4839.7 1533.64  4844.8 1532.75
  4873.3 1532.75  4992.3 1525.39  4995.1 1524.89  4998.3 1525.39  5025.8 1526.49
  5086.8 1525.97  5145.6 1529.01  5168.2 1529.18  5262.0 1533.89  5310.0 1538.24
  5315.1 1537.86  5463.0 1545.18  5506.1 1548.00  5524.0 1548.06  5662.1 1555.34
#Mann=10,-1,0
  3761.7    0.05       0  3901.1     0.1       0  4122.6    0.05       0
  4253.6     0.1       0  4402.9    0.05       0  4571.4     0.1       0
  4770.5    0.16       0  4992.3    0.07       0  4998.3    0.16       0
  5506.1     0.1       0
Bank Sta=4992.3,4998.3
Exp/Cntr=0.3,0.1

Type RM Length L Ch R = 1,18682,491,491,491
BEGIN DESCRIPTION:
UNT007 IN SNOGR 31.0
END DESCRIPTION:
XS GIS Cut Line= 3
      2828370.58     10042608.51      2829770.27     10042738.71
      2830312.79     10042445.75
#Sta/Elev= 30
  3807.9 1552.14  3906.2 1548.14  3919.8 1548.22  4024.0 1544.36  4138.2 1541.06
  4197.5 1538.30  4217.6 1538.36  4307.9 1535.57  4455.8 1533.38  4468.6 1532.03
  4699.6 1525.68  4729.8 1524.23  4783.5 1523.68  4810.1 1522.50  4820.1 1523.22
  4865.4 1523.76  4920.6 1523.28  4970.8 1521.72  4998.9 1517.60  5001.7 1517.10
  5004.9 1517.60  5021.0 1522.10  5061.2 1526.62  5091.3 1527.62  5104.2 1527.26
  5259.2 1530.81  5461.0 1538.05  5511.7 1540.60  5533.0 1541.33  5830.2 1553.28
#Mann=7,-1,0
  3807.9     0.1       0  4865.4    0.16       0  4998.9    0.07       0
  5004.9    0.16       0  5104.2     0.1       0  5511.7    0.16       0
  5533.0     0.1       0
Bank Sta=4998.9,5004.9
Exp/Cntr=0.3,0.1

Type RM Length L Ch R = 1,18191,438,438,438
BEGIN DESCRIPTION:
UNT007 IN SNOGR 30.0
END DESCRIPTION:
XS GIS Cut Line= 4
      2828348.84     10042825.52      2829477.30     10043129.34
      2829770.27     10043053.38      2830388.74     10042543.42
#Sta/Elev= 30
  4049.2 1552.86  4097.4 1551.05  4205.6 1547.37  4406.9 1541.22  4514.8 1539.38
  4521.6 1538.38  4561.5 1535.98  4716.1 1527.98  4750.9 1524.90  4812.1 1521.42
  4846.2 1520.27  4960.1 1519.45  4998.6 1514.96  5001.3 1514.46  5004.6 1514.96
  5020.2 1517.13  5084.4 1517.79  5100.0 1519.23  5115.1 1519.56  5174.8 1520.52
  5286.8 1520.89  5526.5 1524.44  5527.2 1524.45  5674.2 1527.59  5831.8 1532.15
  5844.9 1532.52  6086.6 1541.16  6172.5 1544.98  6189.7 1545.16  6322.1 1550.50
#Mann=15,-1,0
  4049.2     0.1       0  4097.4    0.05       0  4205.6     0.1       0
  4812.1    0.16       0  4998.6    0.07       0  5004.6    0.16       0
  5115.1     0.1       0  5286.8    0.16       0  5526.5     0.1       0
  5527.2    0.16       0  5674.2     0.1       0  5831.8    0.16       0
  5844.9     0.1       0  6086.6    0.16       0  6189.7     0.1       0
Bank Sta=4998.6,5004.6
Exp/Cntr=0.3,0.1

Type RM Length L Ch R = 1,17753,682,682,682
BEGIN DESCRIPTION:
Mapping XS 8dd9c879
END DESCRIPTION:
XS GIS Cut Line= 3
      2827922.89     10043112.84      2829040.90     10043515.60
      2830679.78     10042730.89
#Sta/Elev= 30
  3602.2 1548.09  3764.7 1545.70  4004.9 1539.93  4309.6 1535.95  4511.6 1534.84
  4543.5 1532.71  4617.7 1531.27  4653.7 1528.15  4684.4 1529.35  4711.8 1527.24
  4769.7 1524.07  4803.8 1522.31  4856.3 1520.79  4873.5 1519.24  4954.2 1517.92
  4969.7 1516.32  4995.5 1511.94  4998.2 1511.44  5001.5 1511.94  5009.5 1512.91
  5015.0 1514.93  5053.9 1514.29  5111.2 1516.67  5210.6 1516.33  5457.6 1520.17
  5548.0 1521.95  6064.4 1533.00  6380.8 1540.70  6520.9 1543.31  6607.6 1545.32
#Mann=12,-1,0
  3602.2     0.1       0  4711.8    0.16       0  4769.7    0.05       0
  4803.8    0.16       0  4995.5    0.07       0  5001.5    0.16       0
  5210.6     0.1       0  5457.6    0.16       0  5548.0     0.1       0
  6064.4    0.16       0  6380.8     0.1       0  6520.9    0.16       0
Bank Sta=4995.5,5001.5
Exp/Cntr=0.3,0.1

Type RM Length L Ch R = 1,17071,329,329,329
BEGIN DESCRIPTION:
UNT007 IN SNOGR 29.0
END DESCRIPTION:
XS GIS Cut Line= 2
      2828750.26     10043812.93      2830421.33     10043823.78
#Sta/Elev= 30
  4081.7 1526.52  4269.9 1523.67  4349.9 1521.01  4389.9 1518.62  4429.9 1518.97
  4469.9 1516.60  4599.9 1513.38  4719.9 1512.44  4789.9 1511.44  4839.9 1511.94
  4849.9 1511.19  4876.0 1510.78  4969.9 1509.56  4980.1 1509.11  4996.9 1505.72
  4999.7 1505.22  5002.9 1505.72  5008.3 1507.46  5009.9 1507.98  5040.2 1511.32
  5059.9 1513.35  5139.9 1518.07  5189.9 1518.59  5202.8 1519.08  5229.9 1520.82
  5335.1 1524.18  5529.9 1530.73  5579.9 1531.86  5649.9 1534.44  5752.8 1536.73
#Mann=8,-1,0
  4081.7    0.05       0  4876.0     0.1       0  4996.9    0.07       0
  5002.9     0.1       0  5008.3    0.16       0  5040.2     0.1       0
  5202.8    0.16       0  5335.1     0.1       0
Bank Sta=4996.9,5002.9
Exp/Cntr=0.3,0.1

Type RM Length L Ch R = 1,16742,387,387,387
BEGIN DESCRIPTION:
UNT007 IN SNOGR 28.0
END DESCRIPTION:
XS GIS Cut Line= 3
      2828728.57     10043921.43      2829477.30     10044149.30
      2830312.82     10044116.75
#Sta/Elev= 30
  4059.3 1523.78  4183.4 1522.15  4268.3 1519.99  4325.3 1519.84  4467.1 1513.68
  4598.5 1510.86  4707.6 1509.41  4794.8 1509.12  4811.8 1508.90  4841.0 1507.34
  4895.1 1506.90  4983.2 1507.73  4994.0 1505.15  5000.2 1504.96  5003.0 1504.46
  5006.2 1504.96  5013.2 1506.64  5023.2 1507.32  5043.3 1508.03  5093.3 1508.49
  5110.9 1509.77  5115.9 1509.67  5145.9 1512.73  5193.4 1516.41  5243.4 1521.67
  5303.5 1526.81  5488.5 1530.58  5573.7 1531.55  5593.7 1532.51  5678.1 1534.04
#Mann=8,-1,0
  4059.3    0.05       0  4794.8     0.1       0  4895.1    0.05       0
  4994.0     0.1       0  5000.2    0.07       0  5006.2     0.1       0
  5145.9    0.05       0  5488.5    0.16       0
Bank Sta=5000.2,5006.2
Exp/Cntr=0.3,0.1

Type RM Length L Ch R = 1,16355,360,360,360
BEGIN DESCRIPTION:
Mapping XS 3f8f0f48
END DESCRIPTION:
XS GIS Cut Line= 3
      2828555.00     10044160.15      2829759.42     10044550.78
      2830312.81     10044333.76
#Sta/Elev= 30
  4074.7 1521.63  4103.6 1522.40  4141.4 1520.45  4194.0 1518.96  4359.4 1516.97
  4551.2 1512.51  4711.0 1509.93  4785.6 1507.86  4803.7 1508.23  4856.3 1507.31
  4881.5 1507.86  4919.4 1506.39  4977.4 1505.67  5000.5 1501.07  5003.2 1500.57
  5006.5 1501.07  5009.4 1503.86  5024.5 1505.19  5085.4 1505.34  5187.7 1505.19
  5334.4 1507.51  5429.9 1509.89  5538.4 1514.61  5573.4 1518.38  5617.1 1523.20
  5640.6 1525.00  5718.4 1525.48  5826.2 1527.44  5934.0 1529.71  5935.3 1529.71
#Mann=10,-1,0
  4074.7    0.05       0  4711.0     0.1       0  5000.5    0.07       0
  5006.5     0.1       0  5085.4    0.16       0  5187.7    0.05       0
  5573.4     0.1       0  5718.4    0.05       0  5826.2    0.16       0
  5934.0    0.05       0
Bank Sta=5000.5,5006.5
Exp/Cntr=0.3,0.1

Type RM Length L Ch R = 1,15995,506,506,506
BEGIN DESCRIPTION:
UNT007 IN SNOGR 27.0
END DESCRIPTION:
XS GIS Cut Line= 3
      2828522.45     10044561.63      2829292.84     10044767.79
      2830193.47     10044756.94
#Sta/Elev= 30
  4094.9 1518.14  4124.7 1518.00  4199.6 1515.18  4256.6 1514.11  4394.7 1512.53
  4437.6 1511.14  4622.8 1508.95  4867.2 1505.20  4908.0 1505.61  4928.0 1504.28
  4978.0 1503.10  4995.0 1498.93  4997.8 1498.43  5001.0 1498.93  5018.0 1502.42
  5048.0 1503.31  5098.0 1502.85  5158.0 1501.18  5204.4 1502.17  5277.4 1503.94
  5368.1 1506.68  5418.1 1511.90  5478.1 1516.53  5498.1 1517.04  5528.1 1516.62
  5558.1 1517.29  5618.1 1517.19  5643.7 1519.08  5668.1 1518.21  5793.1 1518.37
#Mann=8,-1,0
  4094.9    0.05       0  4256.6     0.1       0  4437.6    0.05       0
  4622.8     0.1       0  4995.0    0.07       0  5001.0     0.1       0
  5204.4    0.05       0  5277.4     0.1       0
Bank Sta=4995,5001
Exp/Cntr=0.3,0.1

Type RM Length L Ch R = 1,15489,484,484,484
BEGIN DESCRIPTION:
UNT007 IN SNOGR 26.0
END DESCRIPTION:
XS GIS Cut Line= 4
      2828218.58     10044691.82      2829206.04     10045125.86
      2830074.09     10045093.31      2830388.75     10044865.46
#Sta/Elev= 30
  3448.1 1523.77  3480.7 1523.80  3600.9 1518.39  3738.0 1514.75  4386.0 1504.66
  4518.5 1503.16  4589.2 1503.56  4629.9 1501.38  4699.3 1499.41  4779.4 1498.50
  4799.4 1499.51  4908.4 1499.67  4969.0 1498.91  4984.2 1499.12  4996.5 1495.94
  4999.3 1495.44  5002.5 1495.94  5019.5 1499.15  5039.5 1501.05  5163.5 1504.09
  5252.7 1506.94  5259.7 1506.27  5279.7 1508.18  5299.7 1508.83  5339.7 1509.44
  5404.9 1508.64  5499.5 1510.34  5620.9 1514.49  5656.4 1513.79  5783.9 1518.47
#Mann=9,-1,0
  3448.1    0.05       0  4386.0     0.1       0  4629.9    0.05       0
  4908.4     0.1       0  4969.0    0.05       0  4996.5   0.035       0
  5002.5    0.05       0  5163.5     0.1       0  5404.9    0.05       0
Bank Sta=4996.5,5002.5
Exp/Cntr=0.3,0.1

Type RM Length L Ch R = 1,15005,97,97,97
BEGIN DESCRIPTION:
UNT007 IN SNOGR 25.0
END DESCRIPTION:
XS GIS Cut Line= 3
      2828730.61     10045165.89      2829492.32     10045437.16
      2830414.05     10045434.99
#Sta/Elev= 30
  4290.5 1508.43  4500.5 1506.73  4600.5 1504.91  4638.6 1503.94  4711.9 1502.52
  4752.2 1502.27  4829.6 1500.98  4866.0 1500.93  4935.8 1497.49  4984.0 1496.60
  4996.4 1495.33  4999.2 1494.83  5002.4 1495.33  5014.9 1497.14  5071.2 1496.27
  5114.4 1497.32  5155.2 1496.34  5195.2 1496.73  5275.2 1496.03  5325.2 1497.52
  5377.5 1497.84  5476.2 1498.89  5575.2 1501.27  5675.2 1500.51  5745.2 1501.83
  5805.2 1503.31  5855.2 1506.08  5911.5 1508.09  5942.2 1508.62  6020.8 1511.62
#Mann=11,-1,0
  4290.5    0.05       0  4600.5     0.1       0  4638.6    0.05       0
  4752.2     0.1       0  4996.4    0.07       0  5002.4     0.1       0
  5114.4    0.05       0  5377.5     0.1       0  5476.2    0.05       0
  5911.5     0.1       0  5942.2    0.05       0
Bank Sta=4996.4,5002.4
Exp/Cntr=0.3,0.1

Type RM Length L Ch R = 1,14908,177,177,177
BEGIN DESCRIPTION:
Mapping XS 98d2ce23
END DESCRIPTION:
XS GIS Cut Line= 2
      2828706.94     10045483.94      2830334.01     10045510.81
#Sta/Elev= 30
  4335.8 1506.25  4567.4 1506.12  4617.4 1505.68  4706.8 1504.06  4787.4 1502.97
  4837.4 1502.93  4897.4 1498.67  4947.4 1497.94  4997.4 1495.02  5007.4 1495.75
  5037.4 1496.46  5117.1 1496.42  5187.4 1495.09  5227.0 1495.54  5264.5 1494.50
  5267.2 1494.00  5270.5 1494.50  5287.5 1495.01  5327.5 1495.13  5357.5 1496.64
  5377.5 1497.17  5397.0 1497.18  5495.6 1498.09  5717.5 1500.84  5777.5 1502.90
  5834.8 1505.66  5887.5 1506.59  5916.6 1508.29  5937.5 1509.16  5963.1 1509.44
#Mann=8,-1,0
  4335.8    0.05       0  4706.8     0.1       0  5117.1    0.05       0
  5264.5    0.07       0  5270.5    0.05       0  5397.0     0.1       0
  5495.6    0.05       0  5916.6     0.1       0
Bank Sta=5264.5,5270.5
Exp/Cntr=0.3,0.1

Type RM Length L Ch R = 1,14731,613,613,613
BEGIN DESCRIPTION:
Mapping XS ea6c6b66
END DESCRIPTION:
XS GIS Cut Line= 2
      2828685.25     10045635.85      2830334.04     10045630.62
#Sta/Elev= 30
  4217.7 1506.30  4330.9 1506.34  4470.9 1505.64  4580.9 1504.58  4660.9 1503.35
  4760.9 1501.04  4910.9 1498.83  4950.9 1496.30  4970.9 1495.45  4987.0 1493.77
  5000.9 1492.82  5030.9 1493.90  5050.9 1492.55  5067.9 1492.25  5070.7 1491.75
  5073.9 1492.25  5100.9 1493.89  5196.1 1493.25  5230.9 1493.17  5250.9 1492.48
  5294.8 1492.94  5330.9 1493.59  5393.5 1495.54  5420.9 1496.14  5450.9 1496.14
  5520.9 1499.16  5690.9 1503.31  5805.5 1506.78  5840.9 1508.18  5866.5 1509.70
#Mann=8,-1,0
  4217.7    0.05       0  4987.0     0.1       0  5067.9    0.07       0
  5073.9     0.1       0  5196.1    0.05       0  5294.8     0.1       0
  5393.5    0.05       0  5805.5     0.1       0
Bank Sta=5067.9,5073.9
Exp/Cntr=0.3,0.1

Type RM Length L Ch R = 1,14118,471,471,471
BEGIN DESCRIPTION:
UNT007 IN SNOGR 24.0
END DESCRIPTION:
XS GIS Cut Line= 2
      2828815.42     10045863.71      2830271.39     10045940.63
#Sta/Elev= 30
  3994.4 1505.19  4077.6 1504.65  4137.6 1503.76  4247.8 1501.92  4297.9 1500.50
  4368.0 1499.44  4398.0 1498.58  4508.2 1496.80  4523.4 1497.05  4660.8 1492.88
  4698.4 1492.47  4718.5 1492.94  4738.5 1492.27  4850.2 1490.92  4890.1 1490.89
  4978.8 1490.68  4988.8 1490.35  4995.8 1488.07  4998.6 1487.57  5001.8 1488.07
  5018.9 1490.50  5035.6 1491.94  5040.6 1491.19  5058.9 1492.96  5079.0 1492.97
  5129.0 1495.45  5259.2 1497.25  5309.3 1499.04  5415.5 1504.30  5452.4 1505.68
#Mann=6,-1,0
  3994.4    0.05       0  4523.4     0.1       0  4850.2    0.05       0
  4890.1     0.1       0  4995.8    0.07       0  5001.8     0.1       0
Bank Sta=4995.8,5001.8
Exp/Cntr=0.3,0.1

Type RM Length L Ch R = 1,13647,436,436,436
BEGIN DESCRIPTION:
UNT007 IN SNOGR 23.0
END DESCRIPTION:
XS GIS Cut Line= 3
      2828962.84     10045960.17      2829616.02     10046235.77
      2830369.04     10046114.24
#Sta/Elev= 30
  4381.5 1502.79  4420.2 1502.12  4463.6 1500.74  4496.1 1500.36  4572.1 1498.11
  4615.5 1497.66  4691.7 1495.87  4769.6 1495.07  4778.3 1495.16  4810.3 1493.72
  4916.0 1490.90  4974.3 1487.97  4992.6 1487.88  4995.0 1487.24  4997.8 1486.74
  5001.0 1487.24  5016.3 1488.22  5045.4 1488.64  5074.6 1488.43  5193.2 1488.94
  5260.1 1490.39  5388.7 1491.51  5538.6 1494.43  5574.0 1495.52  5635.8 1498.91
  5640.8 1498.81  5670.3 1500.42  5702.6 1501.60  5781.7 1505.74  5853.2 1508.80
#Mann=4,-1,0
  4381.5    0.05       0  4769.6     0.1       0  4995.0    0.07       0
  5001.0     0.1       0
Bank Sta=4995,5001
Exp/Cntr=0.3,0.1

Type RM Length L Ch R = 1,13211,437,437,437
BEGIN DESCRIPTION:
UNT007 IN SNOGR 22.0
END DESCRIPTION:
XS GIS Cut Line= 2
      2829021.59     10046373.70      2830074.86     10046655.44
#Sta/Elev= 30
  4325.7 1499.84  4421.7 1497.71  4426.9 1497.97  4529.5 1495.47  4598.5 1494.63
  4616.8 1494.45  4633.0 1493.18  4651.7 1492.21  4656.8 1492.33  4715.8 1488.37
  4777.9 1486.23  4860.7 1486.08  4886.8 1486.42  4953.9 1485.95  4985.0 1485.39
  4995.3 1484.51  4998.8 1482.83  5001.5 1482.33  5004.8 1482.83  5016.0 1486.12
  5026.4 1487.54  5036.7 1487.85  5212.7 1490.48  5271.8 1491.88  5277.0 1491.52
  5305.9 1492.31  5326.6 1492.13  5351.9 1492.60  5386.8 1494.31  5416.0 1495.12
#Mann=4,-1,0
  4325.7    0.05       0  4598.5     0.1       0  4998.8    0.07       0
  5004.8     0.1       0
Bank Sta=4998.8,5004.8
Exp/Cntr=0.3,0.1

Type RM Length L Ch R = 1,12774,541,541,541
BEGIN DESCRIPTION:
UNT007 IN SNOGR 21.0
END DESCRIPTION:
XS GIS Cut Line= 2
      2829056.15     10046628.57      2830124.72     10047007.88
#Sta/Elev= 30
  4720.5 1498.96  4781.0 1498.34  4947.3 1494.14  4955.6 1493.05  4960.9 1493.14
  4977.6 1486.51  4986.5 1482.19  4991.8 1480.52  4995.9 1480.16  4998.6 1479.66
  5001.9 1480.16  5009.5 1481.73  5017.3 1482.36  5048.2 1483.39  5053.5 1482.98
  5079.1 1484.55  5104.6 1484.46  5109.9 1483.86  5171.7 1483.94  5197.2 1484.89
  5391.5 1485.85  5464.4 1486.82  5469.7 1486.47  5534.7 1487.76  5635.5 1490.85
  5723.0 1494.56  5762.4 1496.82  5767.7 1496.50  5798.6 1497.73  5854.4 1500.95
#Mann=6,-1,0
  4720.5    0.05       0  4947.3     0.1       0  4995.9    0.07       0
  5001.9     0.1       0  5534.7    0.05       0  5723.0     0.1       0
Bank Sta=4995.9,5001.9
Exp/Cntr=0.3,0.1

Type RM Length L Ch R = 1,12233,352,352,352
BEGIN DESCRIPTION:
UNT007 IN SNOGR 20.0
END DESCRIPTION:
XS GIS Cut Line= 2
      2829047.48     10046964.95      2829955.05     10047253.03
#Sta/Elev= 30
  4458.8 1494.43  4575.5 1490.51  4643.8 1488.76  4659.2 1488.65  4699.3 1486.54
  4724.1 1485.66  4795.6 1482.06  4806.6 1482.13  4827.0 1481.59  4838.8 1481.59
  4890.0 1480.26  4898.1 1480.48  4935.6 1480.02  4962.6 1479.10  4967.9 1478.67
  4984.4 1478.82  4991.9 1478.16  4994.7 1477.66  4997.9 1478.16  5005.4 1478.18
  5015.9 1480.43  5026.4 1482.17  5032.4 1482.60  5037.1 1482.32  5057.9 1483.16
  5129.2 1484.00  5134.5 1483.87  5199.0 1485.49  5288.7 1489.29  5411.0 1495.82
#Mann=6,-1,0
  4458.8    0.05       0  4643.8     0.1       0  4724.1    0.05       0
  4991.9   0.035       0  4997.9    0.05       0  5037.1     0.1       0
Bank Sta=4991.9,4997.9
Exp/Cntr=0.3,0.1

Type RM Length L Ch R = 1,11881,240,240,240
BEGIN DESCRIPTION:
UNT007 IN SNOGR 19.0
END DESCRIPTION:
XS GIS Cut Line= 3
      2828934.63     10047108.19      2829366.45     10047379.43
      2829891.61     10047440.19
#Sta/Elev= 30
  4579.9 1494.29  4664.3 1492.49  4774.1 1488.73  4877.7 1486.46  4898.9 1485.15
  4904.9 1483.40  4935.5 1481.90  4962.6 1478.53  4972.0 1477.79  4996.1 1473.49
  4998.8 1472.99  5002.1 1473.49  5035.6 1477.85  5050.9 1478.86  5122.1 1480.96
  5196.8 1480.62  5283.1 1480.09  5346.7 1481.04  5400.6 1483.22  5430.4 1484.59
  5435.5 1484.14  5464.3 1486.89  5494.5 1489.01  5519.3 1490.24  5554.9 1493.36
  5595.2 1494.46  5603.0 1495.38  5608.1 1493.90  5614.4 1495.28  5618.5 1495.28
#Mann=6,-1,0
  4579.9    0.05       0  4664.3     0.1       0  4996.1    0.07       0
  5002.1     0.1       0  5196.8    0.05       0  5400.6     0.1       0
Bank Sta=4996.1,5002.1
Exp/Cntr=0.3,0.1

Type RM Length L Ch R = 1,11641,404,404,404
BEGIN DESCRIPTION:
UNT007 IN SNOGR 18.0
END DESCRIPTION:
XS GIS Cut Line= 3
      2828856.49     10047279.62      2829149.44     10047500.96
      2829791.75     10047529.17
#Sta/Elev= 30
  4590.6 1492.70  4602.5 1492.88  4645.8 1491.53  4680.8 1489.31  4702.4 1488.49
  4730.9 1486.42  4752.4 1485.63  4773.2 1483.61  4794.0 1480.49  4808.6 1479.04
  4844.0 1476.78  4858.5 1476.27  4930.0 1476.03  4976.8 1476.03  5003.8 1475.13
  5006.6 1474.63  5009.8 1475.13  5016.9 1475.92  5026.9 1476.35  5106.9 1477.30
  5127.0 1478.76  5133.5 1479.61  5147.0 1480.18  5257.1 1479.17  5317.1 1479.30
  5407.2 1480.25  5506.9 1484.82  5517.3 1485.13  5586.6 1490.20  5600.7 1490.74
#Mann=6,-1,0
  4590.6    0.05       0  4645.8     0.1       0  4930.0    0.05       0
  5003.8   0.035       0  5009.8    0.05       0  5506.9     0.1       0
Bank Sta=5003.8,5009.8
Exp/Cntr=0.3,0.1

Type RM Length L Ch R = 1,11237,109,109,109
BEGIN DESCRIPTION:
Mapping XS 31e8761e
END DESCRIPTION:
XS GIS Cut Line= 2
      2828680.72     10047566.06      2829754.98     10047557.71
#Sta/Elev= 30
  4755.3 1490.43  4783.1 1489.61  4901.7 1487.94  4923.1 1487.89  4953.1 1484.94
  4963.1 1482.94  4973.1 1480.13  4983.1 1476.74  4990.1 1473.25  4992.8 1472.75
  4996.1 1473.25  5003.1 1473.44  5013.1 1474.58  5053.1 1474.78  5093.1 1474.29
  5133.1 1474.76  5173.1 1475.68  5233.1 1478.55  5283.1 1479.60  5313.1 1479.07
  5373.1 1479.73  5413.1 1479.21  5493.1 1479.35  5521.6 1478.91  5683.1 1480.59
  5733.1 1482.55  5779.5 1485.12  5793.1 1485.81  5813.1 1487.88  5829.6 1488.89
#Mann=6,-1,0
  4755.3    0.05       0  4901.7     0.1       0  4990.1    0.07       0
  4996.1     0.1       0  5521.6    0.05       0  5779.5     0.1       0
Bank Sta=4990.1,4996.1
Exp/Cntr=0.3,0.1

Type RM Length L Ch R = 1,11128,321,321,321
BEGIN DESCRIPTION:
Mapping XS 6d641f23
END DESCRIPTION:
XS GIS Cut Line= 2
      2828713.28     10047646.36      2829693.76     10047651.45
#Sta/Elev= 30
  4719.6 1488.93  4724.8 1488.52  4764.8 1487.89  4842.8 1487.09  4864.8 1486.37
  4894.8 1485.96  4924.8 1483.87  4944.8 1481.54  4954.8 1479.82  4964.8 1476.80
  4984.8 1472.43  4994.8 1471.32  5001.8 1471.09  5004.5 1470.59  5007.8 1471.09
  5024.8 1472.78  5084.8 1474.62  5124.8 1475.19  5134.8 1476.03  5184.8 1478.39
  5244.8 1478.57  5254.8 1479.07  5314.8 1478.42  5444.8 1479.34  5474.8 1479.31
  5504.8 1478.66  5564.8 1478.56  5644.8 1479.86  5684.8 1481.81  5700.1 1483.70
#Mann=4,-1,0
  4719.6    0.05       0  4842.8     0.1       0  5001.8    0.07       0
  5007.8     0.1       0
Bank Sta=5001.8,5007.8
Exp/Cntr=0.3,0.1

Type RM Length L Ch R = 1,10807,280,280,280
BEGIN DESCRIPTION:
UNT007 IN SNOGR 17.0
END DESCRIPTION:
XS GIS Cut Line= 3
      2828855.16     10047918.49      2829153.34     10047891.15
      2829750.07     10047688.31
#Sta/Elev= 30
  4640.1 1482.19  4640.5 1482.19  4659.5 1481.96  4723.8 1480.87  4742.9 1481.02
  4824.2 1478.91  4857.9 1476.74  4904.5 1472.65  4939.5 1471.27  4966.1 1469.42
  4974.7 1469.31  4980.0 1469.89  4987.2 1469.34  4994.8 1467.91  4997.5 1467.41
  5000.8 1467.91  5006.1 1468.78  5018.9 1474.59  5029.4 1475.82  5089.4 1476.65
  5177.3 1476.40  5187.9 1476.94  5251.2 1477.17  5288.5 1476.73  5314.6 1477.22
  5345.8 1476.45  5382.7 1476.54  5462.5 1479.23  5534.3 1483.52  5569.8 1487.02
#Mann=7,-1,0
  4640.1     0.1       0  4640.5    0.16       0  4659.5     0.1       0
  4994.8    0.07       0  5000.8     0.1       0  5089.4    0.16       0
  5345.8    0.05       0
Bank Sta=4994.8,5000.8
Exp/Cntr=0.3,0.1

Type RM Length L Ch R = 1,10527,388,388,388
BEGIN DESCRIPTION:
UNT007 IN SNOGR 16.0
END DESCRIPTION:
XS GIS Cut Line= 3
      2828926.81     10048194.53      2829504.90     10048059.12
      2829853.65     10047845.71
#Sta/Elev= 30
  4702.3 1478.54  4776.3 1478.52  4859.8 1477.21  4888.9 1476.92  4916.6 1475.88
  4940.2 1475.01  4960.8 1473.39  4971.0 1471.52  4988.6 1467.27  4993.8 1465.37
  4998.9 1464.47  5001.6 1463.97  5004.9 1464.47  5031.1 1469.12  5042.9 1470.37
  5078.7 1471.52  5123.7 1471.68  5186.7 1473.84  5258.8 1474.22  5279.2 1473.84
  5301.4 1474.33  5323.7 1474.03  5347.1 1474.89  5369.1 1474.44  5411.7 1475.79
  5478.4 1477.06  5527.8 1478.05  5564.5 1479.68  5638.0 1481.49  5704.9 1484.01
#Mann=7,-1,0
  4702.3     0.1       0  4859.8    0.16       0  4916.6     0.1       0
  4998.9    0.07       0  5004.9     0.1       0  5123.7    0.16       0
  5478.4    0.05       0
Bank Sta=4998.9,5004.9
Exp/Cntr=0.3,0.1

Type RM Length L Ch R = 1,10139,341,341,341
BEGIN DESCRIPTION:
UNT007 IN SNOGR 15.0
END DESCRIPTION:
XS GIS Cut Line= 3
      2829010.14     10048395.92      2829520.53     10048399.39
      2830007.47     10048198.38
#Sta/Elev= 30
  4590.7 1476.70  4639.0 1476.81  4699.0 1475.80  4839.0 1471.21  4889.0 1470.30
  4919.0 1468.74  4939.0 1468.37  4949.0 1467.54  4959.0 1467.79  4969.0 1467.43
  4979.0 1466.75  4989.0 1465.17  4998.9 1461.60  5000.9 1461.43  5003.6 1460.93
  5006.9 1461.43  5009.0 1463.45  5019.0 1464.70  5039.0 1469.09  5059.0 1471.18
  5097.6 1472.23  5132.9 1471.95  5186.1 1472.57  5204.7 1471.84  5236.0 1471.89
  5272.0 1472.37  5369.8 1474.75  5510.0 1476.27  5548.1 1478.01  5627.9 1480.52
#Mann=4,-1,0
  4590.7    0.16       0  5000.9    0.07       0  5006.9    0.16       0
  5236.0    0.05       0
Bank Sta=5000.9,5006.9
Exp/Cntr=0.3,0.1

Type RM Length L Ch R = 1,9798,234,234,234
BEGIN DESCRIPTION:
Mapping XS 925ec11e
END DESCRIPTION:
XS GIS Cut Line= 2
      2829096.89     10048823.02      2830027.46     10048533.08
#Sta/Elev= 30
  4679.6 1472.22  4687.8 1472.13  4712.7 1471.84  4760.5 1469.67  4821.0 1469.17
  4953.6 1468.46  4966.1 1467.76  4974.5 1465.52  4985.0 1463.57  4993.4 1461.18
  4995.6 1459.81  4998.4 1459.31  5001.6 1459.81  5006.0 1460.55  5016.4 1463.48
  5058.3 1465.06  5089.7 1466.83  5128.7 1467.72  5161.2 1467.14  5184.0 1467.34
  5193.8 1467.08  5264.0 1468.22  5288.8 1467.54  5344.8 1468.46  5404.6 1469.17
  5431.9 1468.88  5469.6 1470.49  5540.1 1472.51  5592.5 1474.66  5654.3 1475.80
#Mann=6,-1,0
  4679.6    0.16       0  4687.8     0.1       0  4821.0    0.16       0
  4995.6    0.07       0  5001.6    0.16       0  5344.8    0.05       0
Bank Sta=4995.6,5001.6
Exp/Cntr=0.3,0.1

Type RM Length L Ch R = 1,9564,305,305,305
BEGIN DESCRIPTION:
UNT007 IN SNOGR 14.0
END DESCRIPTION:
XS GIS Cut Line= 2
      2829162.69     10049031.67      2830058.70     10048715.38
#Sta/Elev= 30
  4587.3 1470.99  4628.4 1471.67  4650.2 1471.27  4690.2 1472.01  4721.1 1472.00
  4741.5 1471.41  4777.7 1471.75  4803.3 1470.09  4834.2 1468.94  4862.7 1468.67
  4896.1 1468.36  4927.0 1466.59  4968.9 1462.10  4983.6 1461.38  4988.9 1460.69
  4993.4 1459.33  4996.2 1458.83  4999.4 1459.33  5007.0 1459.33  5019.8 1462.52
  5050.7 1463.54  5107.3 1463.12  5132.9 1463.91  5144.9 1464.96  5287.7 1466.80
  5344.1 1467.14  5380.3 1468.92  5452.4 1471.22  5484.2 1473.22  5537.5 1474.44
#Mann=7,-1,0
  4587.3     0.1       0  4650.2    0.16       0  4862.7    0.05       0
  4968.9    0.16       0  4993.4    0.07       0  4999.4    0.16       0
  5287.7    0.05       0
Bank Sta=4993.4,4999.4
Exp/Cntr=0.3,0.1

Type RM Length L Ch R = 1,9259,239,239,239
BEGIN DESCRIPTION:
Mapping XS a4b3a6dd
END DESCRIPTION:
XS GIS Cut Line= 3
      2829246.07     10049151.45      2829709.77     10049071.27
      2830152.44     10048882.05
#Sta/Elev= 30
  4439.5 1469.42  4456.3 1469.30  4472.4 1470.13  4482.5 1470.05  4511.0 1468.98
  4604.3 1467.43  4630.6 1466.40  4711.3 1465.69  4810.0 1464.47  4858.0 1465.06
  4913.3 1463.56  4952.2 1460.12  4984.8 1459.63  5003.5 1457.50  5006.3 1457.00
  5009.5 1457.50  5015.1 1458.17  5022.7 1459.98  5028.3 1461.81  5038.7 1463.48
  5050.0 1464.12  5067.8 1464.34  5091.4 1463.16  5120.4 1463.96  5132.0 1463.77
  5149.4 1463.80  5194.8 1465.63  5267.4 1468.70  5332.8 1472.28  5391.5 1474.05
#Mann=8,-1,0
  4439.5     0.1       0  4711.3    0.05       0  4913.3     0.1       0
  5003.5    0.07       0  5009.5     0.1       0  5022.7    0.16       0
  5132.0     0.1       0  5194.8    0.05       0
Bank Sta=5003.5,5009.5
Exp/Cntr=0.3,0.1

Type RM Length L Ch R = 1,9020,528,528,528
BEGIN DESCRIPTION:
Mapping XS 9e747b4e
END DESCRIPTION:
XS GIS Cut Line= 3
      2829214.76     10049239.99      2829763.58     10049279.60
      2830173.33     10049140.70
#Sta/Elev= 30
  4287.2 1467.44  4311.0 1467.94  4321.0 1468.58  4341.0 1467.69  4429.5 1466.42
  4547.1 1463.54  4591.7 1462.87  4681.7 1462.52  4837.4 1461.12  4901.6 1462.31
  4916.5 1461.94  4927.1 1462.19  4938.3 1461.05  4945.4 1461.32  4964.4 1460.96
  4979.9 1458.97  4990.4 1458.51  4998.1 1457.33  5000.8 1456.83  5004.1 1457.33
  5011.5 1458.73  5021.9 1459.22  5032.7 1458.41  5053.4 1458.49  5096.0 1463.33
  5116.2 1463.86  5191.0 1468.22  5210.4 1468.45  5251.4 1469.83  5270.1 1469.93
#Mann=6,-1,0
  4287.2     0.1       0  4429.5    0.05       0  4945.4     0.1       0
  4998.1    0.07       0  5004.1     0.1       0  5251.4    0.05       0
Bank Sta=4998.1,5004.1
Exp/Cntr=0.3,0.1

Type RM Length L Ch R = 1,8492,352,352,352
BEGIN DESCRIPTION:
Mapping XS d843851c
END DESCRIPTION:
XS GIS Cut Line= 2
      2829336.53     10049319.55      2830193.76     10049803.70
#Sta/Elev= 30
  4248.9 1465.31  4311.3 1463.24  4451.3 1461.59  4526.5 1462.07  4618.8 1459.92
  4699.7 1460.66  4774.8 1457.61  4812.1 1458.09  4839.8 1456.61  4855.7 1456.42
  4905.7 1457.79  4930.9 1457.66  4974.1 1454.50  4979.8 1454.56  4998.5 1451.57
  5001.2 1451.07  5004.5 1451.57  5023.1 1455.06  5039.1 1460.76  5044.8 1460.67
  5055.0 1462.16  5060.7 1461.58  5066.5 1462.72  5076.6 1463.77  5082.4 1463.58
  5098.3 1465.76  5141.6 1468.94  5184.9 1469.55  5206.4 1470.80  5233.4 1471.83
#Mann=6,-1,0
  4248.9    0.05       0  4812.1     0.1       0  4930.9    0.16       0
  4998.5    0.07       0  5004.5    0.16       0  5206.4     0.1       0
Bank Sta=4998.5,5004.5
Exp/Cntr=0.3,0.1

Type RM Length L Ch R = 1,8140,260,260,260
BEGIN DESCRIPTION:
UNT007 IN SNOGR 13.0
END DESCRIPTION:
XS GIS Cut Line= 2
      2829094.98     10049594.14      2829963.82     10050038.54
#Sta/Elev= 30
  4269.6 1462.05  4285.0 1461.85  4301.6 1463.21  4318.2 1463.64  4390.5 1461.36
  4451.5 1460.93  4479.3 1461.42  4546.0 1459.00  4629.2 1459.34  4701.4 1457.19
  4756.5 1457.43  4784.7 1458.41  4851.3 1456.02  4895.7 1456.65  4923.7 1454.95
  4940.2 1454.46  4962.4 1455.51  4979.0 1453.06  4989.4 1450.04  4992.1 1449.54
  4995.4 1450.04  5014.8 1453.34  5032.1 1453.57  5090.0 1455.15  5140.1 1455.47
  5162.3 1457.97  5178.9 1462.30  5201.1 1464.95  5228.9 1463.23  5245.5 1463.45
#Mann=5,-1,0
  4269.6    0.05       0  4923.7     0.1       0  4989.4    0.07       0
  4995.4     0.1       0  5032.1    0.16       0
Bank Sta=4989.4,4995.4
Exp/Cntr=0.3,0.1

Type RM Length L Ch R = 1,7880,681,681,681
BEGIN DESCRIPTION:
UNT007 IN SNOGR 12.0
END DESCRIPTION:
XS GIS Cut Line= 4
      2829017.03     10050678.93      2829638.58     10050171.96
      2829866.02     10050145.92      2830054.36     10050052.61
#Sta/Elev= 30
  4158.6 1464.04  4249.1 1461.05  4305.1 1457.49  4333.8 1456.88  4397.7 1453.16
  4432.9 1453.52  4476.0 1452.78  4504.7 1451.33  4583.0 1454.21  4618.2 1454.62
  4632.5 1453.77  4710.8 1452.75  4888.1 1452.69  4908.9 1453.61  4942.2 1452.34
  4970.6 1452.06  4992.5 1449.59  4997.8 1447.87  5000.6 1447.37  5003.8 1447.87
  5010.9 1448.51  5021.0 1451.64  5081.7 1452.80  5101.5 1452.42  5151.8 1455.41
  5165.9 1454.84  5171.9 1455.95  5188.3 1456.65  5207.4 1456.77  5399.8 1463.92
#Mann=4,-1,0
  4158.6    0.05       0  4942.2    0.16       0  4997.8    0.07       0
  5003.8    0.16       0
Bank Sta=4997.8,5003.8
Exp/Cntr=0.3,0.1

Type RM Length L Ch R = 1,7199,351,351,351
BEGIN DESCRIPTION:
UNT007 IN SNOGR 11.0
END DESCRIPTION:
XS GIS Cut Line= 3
      2829319.13     10050998.36      2829754.90     10050698.01
      2830140.30     10050121.65
#Sta/Elev= 30
  4594.6 1459.05  4618.1 1457.64  4654.5 1456.78  4719.3 1457.01  4812.4 1455.96
  4820.8 1455.46  4841.7 1455.64  4877.5 1454.50  4928.3 1453.83  4943.2 1452.70
  4985.1 1447.65  4993.9 1445.10  5003.7 1443.05  5006.5 1442.55  5009.7 1443.05
  5014.8 1446.56  5016.1 1446.85  5029.7 1449.28  5035.8 1449.71  5056.7 1449.90
  5122.3 1448.96  5179.2 1449.56  5268.6 1449.18  5323.3 1448.93  5482.5 1450.22
  5662.7 1456.21  5770.8 1461.19  5791.8 1462.94  5812.9 1463.44  5817.2 1463.44
#Mann=6,-1,0
  4594.6    0.05       0  5003.7   0.035       0  5009.7    0.05       0
  5016.1    0.16       0  5268.6    0.05       0  5812.9    0.16       0
Bank Sta=5003.7,5009.7
Exp/Cntr=0.3,0.1

Type RM Length L Ch R = 1,6848,367,367,367
BEGIN DESCRIPTION:
Mapping XS 35d33e52
END DESCRIPTION:
XS GIS Cut Line= 4
      2829588.20     10051154.63      2829938.93     10050921.96
      2830004.90     10050724.05      2830239.30     10050220.54
#Sta/Elev= 30
  4465.0 1455.44  4494.5 1455.31  4537.3 1452.53  4573.3 1453.15  4617.8 1450.15
  4675.0 1450.63  4705.1 1449.15  4819.3 1446.86  4855.4 1448.76  4877.5 1447.51
  4931.6 1448.15  4963.3 1447.16  4968.5 1447.56  4978.9 1446.77  4989.4 1444.77
  4991.9 1441.63  4994.6 1441.13  4997.9 1441.63  5010.5 1442.37  5026.5 1447.15
  5042.1 1447.45  5105.9 1446.45  5181.7 1448.60  5216.2 1448.00  5278.1 1448.20
  5347.4 1449.25  5472.8 1452.55  5541.4 1455.25  5587.2 1458.12  5649.9 1460.98
#Mann=5,-1,0
  4465.0    0.05       0  4877.5    0.16       0  4991.9    0.07       0
  4997.9    0.16       0  5278.1    0.05       0
Bank Sta=4991.9,4997.9
Exp/Cntr=0.3,0.1

Type RM Length L Ch R = 1,6481,309,309,309
BEGIN DESCRIPTION:
UNT007 IN SNOGR 10.0
END DESCRIPTION:
XS GIS Cut Line= 3
      2829614.29     10051237.93      2830284.42     10050786.55
      2830390.32     10050310.87
#Sta/Elev= 30
  4088.5 1455.55  4123.3 1455.64  4165.9 1452.88  4202.1 1453.22  4246.2 1450.52
  4282.2 1451.22  4324.2 1448.86  4360.2 1448.52  4390.2 1447.52  4527.6 1445.55
  4565.0 1446.41  4585.1 1447.81  4636.0 1446.51  4648.2 1447.17  4699.0 1446.94
  4780.0 1445.25  4858.0 1445.79  4930.1 1445.10  4936.7 1444.60  4960.8 1445.64
  4980.2 1444.88  4988.6 1441.72  4991.3 1441.22  4994.6 1441.72  5012.1 1442.52
  5040.2 1446.09  5053.0 1446.90  5140.0 1448.75  5261.6 1452.02  5383.8 1457.40
#Mann=6,-1,0
  4088.5    0.05       0  4565.0    0.16       0  4988.6    0.07       0
  4994.6    0.16       0  5040.2     0.1       0  5140.0    0.05       0
Bank Sta=4988.6,4994.6
Exp/Cntr=0.3,0.1

Type RM Length L Ch R = 1,6172,197,197,197
BEGIN DESCRIPTION:
Mapping XS 1c207162
END DESCRIPTION:
XS GIS Cut Line= 4
      2829631.62     10051265.72      2830308.72     10050989.67
      2830471.92     10050921.96      2830739.26     10050574.77
#Sta/Elev= 30
  4210.3 1455.61  4239.3 1455.56  4279.4 1453.08  4314.9 1453.40  4362.4 1450.74
  4401.3 1451.27  4455.3 1448.69  4570.9 1445.87  4714.5 1444.92  4771.1 1446.10
  4779.3 1446.71  4800.9 1444.68  4814.3 1445.61  4833.0 1445.47  4862.4 1443.86
  4945.3 1443.22  4952.1 1444.14  4974.6 1443.39  4995.5 1439.40  4998.2 1438.90
  5001.5 1439.40  5006.2 1439.41  5027.9 1443.08  5063.4 1444.38  5099.4 1446.30
  5203.2 1446.19  5464.0 1449.19  5507.2 1450.47  5542.8 1454.79  5556.4 1454.83
#Mann=6,-1,0
  4210.3    0.05       0  4771.1    0.16       0  4995.5    0.07       0
  5001.5    0.16       0  5063.4     0.1       0  5203.2    0.05       0
Bank Sta=4995.5,5001.5
Exp/Cntr=0.3,0.1

Type RM Length L Ch R = 1,5975,358,358,358
BEGIN DESCRIPTION:
UNT007 IN SNOGR 9.0
END DESCRIPTION:
XS GIS Cut Line= 3
      2829800.08     10051359.45      2830431.99     10051145.92
      2831133.42     10050673.67
#Sta/Elev= 30
  4378.4 1453.05  4418.9 1451.14  4470.4 1451.48  4513.9 1449.09  4690.6 1445.11
  4821.6 1443.80  4847.8 1442.50  4904.5 1441.44  4952.7 1442.26  4957.2 1442.01
  4973.6 1438.08  4978.9 1438.45  4996.5 1435.64  4999.2 1435.14  5002.5 1435.64
  5005.1 1440.21  5010.4 1438.17  5020.6 1441.86  5024.6 1442.10  5146.8 1443.73
  5340.6 1445.89  5397.6 1447.79  5426.9 1447.38  5520.6 1448.51  5592.6 1449.73
  5619.8 1450.97  5643.5 1449.04  5692.1 1451.93  5823.5 1454.95  5891.0 1457.55
#Mann=6,-1,0
  4378.4    0.05       0  4952.7    0.16       0  4996.5    0.07       0
  5002.5    0.16       0  5024.6     0.1       0  5146.8    0.05       0
Bank Sta=4996.5,5002.5
Exp/Cntr=0.3,0.1

Type RM Length L Ch R = 1,5617,261,261,261
BEGIN DESCRIPTION:
Mapping XS 109d7ebd
END DESCRIPTION:
XS GIS Cut Line= 3
      2829855.64     10051508.77      2830475.39     10051441.06
      2830903.83     10050974.46
#Sta/Elev= 30
  4598.3 1452.03  4631.3 1451.40  4681.6 1451.83  4693.7 1451.46  4711.8 1449.94
  4772.2 1448.85  4802.3 1447.66  4882.8 1446.10  4913.0 1446.22  4933.1 1444.25
  4967.6 1442.52  4984.1 1438.42  4993.5 1434.99  5000.5 1434.79  5003.3 1434.29
  5006.5 1434.79  5013.6 1437.95  5023.6 1439.85  5033.7 1440.07  5053.8 1439.74
  5145.4 1441.39  5164.5 1442.04  5194.7 1442.08  5236.1 1441.55  5289.1 1441.75
  5370.5 1441.64  5498.1 1443.35  5731.8 1445.53  5844.6 1448.04  5855.2 1448.83
#Mann=6,-1,0
  4598.3    0.05       0  4984.1    0.16       0  5000.5    0.07       0
  5006.5    0.16       0  5145.4     0.1       0  5289.1    0.05       0
Bank Sta=5000.5,5006.5
Exp/Cntr=0.3,0.1

Type RM Length L Ch R = 1,5356,313,313,313
BEGIN DESCRIPTION:
Mapping XS cc72ae15
END DESCRIPTION:
XS GIS Cut Line= 3
      2829909.38     10051769.19      2830510.11     10051694.53
      2830872.94     10051048.73
#Sta/Elev= 30
  4636.8 1451.49  4686.3 1452.03  4696.3 1451.02  4721.6 1449.83  4787.0 1447.96
  4877.7 1446.78  4897.9 1447.21  4913.8 1445.49  4928.1 1444.00  4948.3 1443.34
  4964.1 1441.62  4969.2 1441.98  4978.5 1440.00  4988.6 1433.87  4995.6 1431.89
  4998.4 1431.39  5001.6 1431.89  5008.7 1435.21  5018.8 1437.38  5059.1 1439.51
  5079.3 1438.83  5119.4 1438.69  5273.4 1438.51  5410.9 1439.31  5506.9 1441.85
  5621.9 1442.94  5697.1 1442.83  5756.4 1444.01  5843.2 1444.41  5982.9 1446.57
#Mann=6,-1,0
  4636.8    0.05       0  4913.8    0.16       0  4995.6    0.07       0
  5001.6    0.16       0  5119.4     0.1       0  5273.4    0.05       0
Bank Sta=4995.6,5001.6
Exp/Cntr=0.3,0.1

Type RM Length L Ch R = 1,5043,258,258,258
BEGIN DESCRIPTION:
UNT007 IN SNOGR 8.0
END DESCRIPTION:
XS GIS Cut Line= 3
      2830009.00     10052309.01      2830629.90     10051781.34
      2830898.75     10051188.15
#Sta/Elev= 30
  4506.4 1450.90  4538.1 1449.65  4573.2 1450.47  4595.2 1449.02  4614.7 1448.40
  4651.2 1447.41  4708.3 1447.23  4736.9 1447.69  4765.5 1446.26  4784.7 1446.29
  4814.9 1446.30  4886.3 1444.56  4942.3 1441.79  4964.3 1441.19  4978.1 1439.26
  4985.1 1436.63  4996.4 1430.76  4999.2 1430.26  5002.4 1430.76  5013.7 1434.75
  5048.8 1437.62  5155.4 1437.16  5329.2 1437.68  5417.4 1439.22  5666.7 1441.37
  5770.1 1445.34  5787.7 1444.47  5810.0 1444.37  5915.9 1445.11  5972.5 1446.18
#Mann=8,-1,0
  4506.4     0.1       0  4614.7    0.05       0  4784.7     0.1       0
  4996.4    0.07       0  5002.4     0.1       0  5329.2    0.05       0
  5810.0     0.1       0  5915.9    0.05       0
Bank Sta=4996.4,5002.4
Exp/Cntr=0.3,0.1

Type RM Length L Ch R = 1,4785,173,173,173
BEGIN DESCRIPTION:
UNT007 IN SNOGR 7.0
END DESCRIPTION:
XS GIS Cut Line= 4
      2829889.67     10052406.68      2830407.51     10052359.78
      2830860.64     10051776.45      2830860.64     10051651.45
#Sta/Elev= 30
  4270.9 1454.69  4289.8 1454.13  4309.9 1454.33  4329.9 1453.14  4390.6 1451.89
  4420.3 1450.37  4440.4 1450.14  4480.5 1448.54  4601.0 1446.69  4671.7 1446.39
  4766.3 1445.87  4867.0 1445.55  4910.4 1443.59  4931.2 1441.25  4945.7 1441.04
  4952.0 1439.98  4960.2 1439.89  4974.7 1438.33  4995.5 1430.02  4998.8 1430.00
  5001.6 1429.50  5004.8 1430.00  5016.3 1434.84  5030.8 1436.58  5038.9 1436.71
  5095.0 1434.99  5159.3 1436.60  5223.6 1437.44  5422.7 1437.61  5654.5 1439.77
#Mann=6,-1,0
  4270.9    0.05       0  4390.6     0.1       0  4671.7    0.05       0
  4766.3     0.1       0  4998.8    0.07       0  5004.8     0.1       0
Bank Sta=4998.8,5004.8
Exp/Cntr=0.3,0.1

Type RM Length L Ch R = 1,4612,310,310,310
BEGIN DESCRIPTION:
UNT007 IN SNOGR 6.0
END DESCRIPTION:
XS GIS Cut Line= 3
      2830182.59     10052732.21      2830834.59     10052161.86
      2831042.92     10051729.60
#Sta/Elev= 30
  4394.4 1444.07  4432.1 1444.40  4602.6 1445.98  4631.1 1445.20  4723.2 1446.14
  4872.2 1445.25  4914.9 1443.59  4943.4 1443.68  4964.3 1440.12  4978.5 1436.73
  4992.7 1431.73  4997.1 1429.17  4999.8 1428.67  5003.1 1429.17  5021.2 1434.10
  5027.8 1435.00  5042.1 1435.74  5064.6 1435.24  5141.7 1433.53  5191.1 1434.27
  5368.6 1434.55  5391.3 1434.50  5396.8 1433.41  5413.9 1433.40  5419.4 1434.84
  5425.1 1435.01  5480.6 1435.31  5555.1 1437.48  5600.4 1437.62  5740.5 1440.55
#Mann=5,-1,0
  4394.4     0.1       0  4432.1    0.05       0  4997.1   0.035       0
  5003.1    0.05       0  5064.6     0.1       0
Bank Sta=4997.1,5003.1
Exp/Cntr=0.3,0.1

Type RM Length L Ch R = 1,4302,365,365,365
BEGIN DESCRIPTION:
Mapping XS 6c919b58
END DESCRIPTION:
XS GIS Cut Line= 2
      2830735.99     10052894.94      2831162.64     10051698.53
#Sta/Elev= 30
  4630.7 1443.99  4717.4 1444.61  4866.1 1444.76  4886.3 1444.56  4891.6 1444.09
  4922.4 1443.19  4939.9 1441.82  4947.9 1440.53  4971.7 1438.24  4984.0 1434.42
  4992.9 1428.80  5000.6 1427.50  5003.3 1427.00  5006.6 1427.50  5009.0 1429.86
  5009.5 1430.35  5014.8 1431.33  5035.0 1433.33  5056.7 1434.48  5111.8 1432.95
  5173.4 1433.02  5216.3 1432.58  5312.3 1431.51  5353.9 1433.08  5399.5 1433.81
  5438.9 1435.57  5481.3 1436.03  5512.1 1436.92  5700.5 1439.29  5900.9 1442.76
#Mann=7,-1,0
  4630.7    0.05       0  5000.6   0.035       0  5006.6    0.05       0
  5009.0     0.1       0  5111.8    0.16       0  5216.3     0.1       0
  5700.5    0.05       0
Bank Sta=5000.6,5006.6
Exp/Cntr=0.3,0.1

Type RM Length L Ch R = 1,3937,323,323,323
BEGIN DESCRIPTION:
Mapping XS 009f63a6
END DESCRIPTION:
XS GIS Cut Line= 4
      2830811.93     10052905.82      2831187.20     10052439.33
      2831114.28     10052284.81      2831173.01     10051777.56
#Sta/Elev= 30
  4338.4 1443.87  4465.7 1443.30  4550.5 1441.92  4579.3 1442.33  4628.9 1439.87
  4643.3 1440.12  4657.7 1439.51  4664.1 1438.60  4672.1 1438.53  4678.5 1437.69
  4771.3 1433.71  4792.8 1433.21  4870.5 1431.79  4954.3 1431.91  4964.6 1431.32
  4976.5 1427.97  4987.3 1427.32  4989.9 1426.51  4992.6 1426.01  4995.9 1426.51
  5010.5 1428.78  5021.2 1430.84  5043.9 1431.01  5089.5 1430.01  5105.8 1431.08
  5149.3 1432.01  5260.0 1436.05  5325.3 1437.68  5378.7 1438.47  5618.6 1441.76
#Mann=8,-1,0
  4338.4    0.05       0  4792.8    0.16       0  4989.9    0.07       0
  4995.9    0.16       0  5010.5     0.1       0  5260.0    0.05       0
  5325.3     0.1       0  5378.7    0.05       0
Bank Sta=4989.9,4995.9
Exp/Cntr=0.3,0.1

Type RM Length L Ch R = 1,3614,525,525,525
BEGIN DESCRIPTION:
Mapping XS 98c5ba28
END DESCRIPTION:
XS GIS Cut Line= 3
      2830844.48     10052949.22      2831451.08     10052300.44
      2831364.28     10051972.32
#Sta/Elev= 30
  4053.7 1442.55  4209.1 1441.95  4251.6 1440.92  4258.5 1441.42  4272.6 1441.40
  4350.3 1437.82  4386.0 1437.28  4435.3 1434.79  4471.0 1434.61  4508.1 1433.40
  4562.8 1431.65  4616.8 1431.83  4676.1 1430.35  4769.7 1429.78  4799.1 1429.92
  4941.9 1429.94  4973.2 1430.46  4979.9 1429.77  4990.2 1425.31  4997.5 1424.63
  5000.3 1424.13  5003.5 1424.63  5008.3 1425.02  5013.4 1427.26  5021.2 1428.05
  5048.5 1429.23  5077.9 1431.35  5104.0 1433.43  5217.8 1436.96  5281.3 1438.32
#Mann=8,-1,0
  4053.7    0.05       0  4508.1    0.16       0  4616.8    0.05       0
  4769.7     0.1       0  4799.1    0.05       0  4997.5   0.035       0
  5003.5    0.05       0  5077.9     0.1       0
Bank Sta=4997.5,5003.5
Exp/Cntr=0.3,0.1

Type RM Length L Ch R = 1,3089,614,614,614
BEGIN DESCRIPTION:
Mapping XS 440869d4
END DESCRIPTION:
XS GIS Cut Line= 4
      2830877.01     10052970.95      2831586.50     10052305.64
      2831713.24     10052345.58      2831900.73     10051972.33
#Sta/Elev= 30
  3965.0 1441.43  4056.0 1441.26  4070.2 1440.49  4119.5 1441.41  4317.8 1434.72
  4346.2 1434.76  4407.7 1433.25  4416.2 1433.15  4438.0 1433.25  4473.6 1431.20
  4629.0 1429.03  4643.2 1427.99  4800.5 1428.77  4890.8 1429.18  4951.7 1427.44
  4971.1 1427.66  4978.8 1427.12  4992.1 1423.00  4999.6 1421.79  5002.3 1421.29
  5005.6 1421.79  5016.4 1426.65  5023.6 1429.00  5034.1 1429.72  5141.0 1429.93
  5158.3 1429.28  5180.6 1429.53  5314.6 1433.07  5320.2 1433.74  5488.2 1436.02
#Mann=7,-1,0
  3965.0    0.05       0  4407.7    0.16       0  4416.2    0.05       0
  4800.5     0.1       0  4999.6    0.07       0  5005.6     0.1       0
  5141.0    0.05       0
Bank Sta=4999.6,5005.6
Exp/Cntr=0.3,0.1

Type RM Length L Ch R = 1,2475,531,531,531
BEGIN DESCRIPTION:
UNT007 IN SNOGR 5.0
END DESCRIPTION:
XS GIS Cut Line= 4
      2830912.92     10053094.69      2831652.47     10052753.56
      2831811.33     10052487.94      2831959.76     10051922.85
#Sta/Elev= 30
  4118.0 1438.61  4130.9 1437.85  4228.2 1437.08  4394.4 1433.69  4422.8 1433.35
  4432.5 1433.86  4445.8 1433.56  4463.2 1432.18  4491.7 1432.00  4606.4 1429.08
  4817.9 1427.91  4936.2 1425.22  4967.2 1425.59  4979.0 1424.37  4988.7 1421.28
  4999.1 1419.73  5001.9 1419.23  5005.1 1419.73  5010.1 1424.25  5025.5 1425.84
  5037.4 1425.39  5068.5 1426.21  5169.6 1426.38  5291.3 1429.61  5308.3 1429.36
  5360.0 1430.49  5372.0 1429.92  5504.8 1431.06  5644.2 1433.28  5826.2 1437.67
#Mann=3,-1,0
  4118.0    0.05       0  4999.1   0.035       0  5005.1    0.05       0
Bank Sta=4999.1,5005.1
Exp/Cntr=0.3,0.1
