HEC-RAS study PEDERNALES RIVER.prj: PEDERNALES RIVER Base Level Engineering

--- PEDERNALES RIVER.g02 (geometry) --- (continued)

Type RM Length L Ch R = 1 ,404954  ,3223,3223,3223
BEGIN DESCRIPTION:
PEDERNALES RIVER 154.0
END DESCRIPTION:
XS GIS Cut Line= 4
      2797663.12     10071589.93       2799535.8     10055824.19
      2797933.69      10038820.2      2795953.64     10030307.92
#Sta/Elev= 30
-18115.3 1693.04-17426.5 1667.47-15460.6 1628.26-14463.6 1614.64-12558.3 1602.45
-10154.4 1592.67   -8352  1585.1 -3154.7 1525.27  -242.4 1523.71    1427 1519.77
  4230.2 1508.77  4300.6 1476.31  4421.1 1493.32  4431.1 1495.46  5043.6 1470.42
    5315 1496.43  5937.3 1488.73  6822.7 1498.84  9776.9 1545.42 11085.1 1567.27
 14524.6 1569.98 16060.8 1562.93 19213.5 1556.06 19621.3 1523.18 19692.4  1548.9
 19937.3 1551.02 22191.4 1583.08 22877.9 1666.08 23192.6 1675.23 23580.1 1669.95
#Mann= 20 ,-1 , 0
-18115.3      .1       0-17426.5     .05       0-15460.6      .1       0
-14463.6      .1       0-12558.3      .1       0-10154.4      .1       0
   -8352      .1       0  -242.4     .05       0    1427      .1       0
  4431.1     .07       0    5315      .1       0  5937.3     .05       0
  6822.7      .1       0  9776.9      .1       0 11085.1      .1       0
 14524.6     .05       0 16060.8     .05       0 19937.3     .05       0
 22191.4     .16       0 23192.6      .1       0
Bank Sta=4421.1,5315
XS Rating Curve= 0 ,0
Exp/Cntr=0.3,0.1

Type RM Length L Ch R = 1 ,401731  ,3308,3308,3308
BEGIN DESCRIPTION:
PEDERNALES RIVER 156.0
END DESCRIPTION:
XS GIS Cut Line= 3
      2800392.65     10072344.35      2801489.62     10053433.16
      2799969.35     10028412.88
#Sta/Elev= 30
-16957.7 1699.31-16165.8 1670.46-14445.3 1677.38-12258.6 1653.92-11492.8 1634.11
 -9564.7 1664.73 -7622.5 1611.86 -5397.7 1624.81 -3996.3 1571.53  1468.2 1504.03
  3598.9 1525.62  4589.5 1491.46  4609.5 1488.31    5000 1455.34  5547.7 1491.86
  5552.7 1491.19  5961.8 1503.61  7020.1 1506.75  7915.2 1508.17  8856.7 1509.66
 13541.3 1535.05 14185.2 1529.39 15722.7  1538.9 17233.1 1527.94 19707.9 1533.03
 20859.5  1506.3 21134.8 1529.78 25659.2 1613.98   27018 1660.86 27051.7 1661.82
#Mann= 20 ,-1 , 0
-16957.7      .1       0-14445.3      .1       0-12258.6      .1       0
-11492.8      .1       0  1468.2      .1       0  3598.9      .1       0
  4609.5     .07       0  5552.7      .1       0  5961.8      .1       0
  7020.1     .05       0  7915.2     .05       0  8856.7     .05       0
 13541.3      .1       0 14185.2     .05       0 15722.7     .05       0
 17233.1     .05       0 19707.9     .05       0 21134.8      .1       0
 25659.2      .1       0   27018     .16       0
Bank Sta=4589.5,5547.7
XS Rating Curve= 0 ,0
Exp/Cntr=0.3,0.1

Type RM Length L Ch R = 1 ,398423  ,1753,1753,1753
BEGIN DESCRIPTION:
PEDERNALES RIVER 157.0
END DESCRIPTION:
XS GIS Cut Line= 4
      2802645.14     10072718.76      2804866.32     10054168.52
      2802541.05     10045459.28      2804895.98     10030208.79
#Sta/Elev= 30
  -16089 1698.46-13790.4 1642.39-12008.6 1649.69-10432.2 1619.46 -9041.5 1578.55
 -8174.3 1591.34 -6939.5 1659.39 -6626.9 1619.55   -6106 1615.71 -4293.5 1608.04
   -2840 1555.01  4689.5 1484.64  4696.4 1483.36  4891.4 1451.12  5343.7 1480.74
  5357.2 1481.95  6384.3    1486  8253.8 1493.38 10519.7 1503.24 14141.4 1513.77
 15551.5 1507.89 17088.9 1498.23 19020.4 1536.09 19131.7 1571.38 20439.4 1612.68
 23315.9 1727.16 24200.6 1656.33 25061.6 1682.73 25776.2 1640.78 27039.3 1664.94
#Mann= 20 ,-1 , 0
  -16089      .1       0-13790.4      .1       0-12008.6      .1       0
-10432.2     .05       0 -9041.5      .1       0 -8174.3      .1       0
   -6106      .1       0 -4293.5      .1       0   -2840      .1       0
  4689.5     .07       0  5343.7      .1       0  5343.7      .1       0
  6384.3     .05       0  8253.8      .1       0 10519.7     .05       0
 14141.4     .05       0 15551.5     .05       0 17088.9     .16       0
 20439.4      .1       0 23315.9      .1       0
Bank Sta=4696.4,5357.2
XS Rating Curve= 0 ,0
Exp/Cntr=0.3,0.1

Type RM Length L Ch R = 1 ,396670  ,2332,2332,2332
BEGIN DESCRIPTION:
PEDERNALES RIVER 163.0
END DESCRIPTION:
XS GIS Cut Line= 3
      2803347.99     10072454.89      2805962.94     10053648.94
      2805338.26     10033544.53
#Sta/Elev= 30
-15426.2 1674.29-14663.7 1660.17-13102.9 1622.52-12412.7 1631.15-10023.6 1631.21
 -9800.7 1613.22 -8405.7  1570.5 -3845.7 1573.09  2718.4 1503.46  4736.5 1486.64
  4831.6 1471.34  4916.3 1450.35  5356.8 1484.94  5452.1 1484.98  7387.7 1485.83
  7717.9 1452.59    7938 1485.94  8703.9  1489.9 10477.7 1519.84 11772.5 1523.67
 12700.1 1523.33 14599.2 1531.82 15498.7 1534.39 16542.2 1531.24 16695.5 1511.02
 18130.4 1539.89 19154.7  1570.9 21170.3 1614.76 23387.4 1728.22 23674.8 1739.72
#Mann= 19 ,-1 , 0
-15426.2      .1       0-14663.7     .16       0-12412.7      .1       0
 -9800.7     .05       0 -8405.7      .1       0  2718.4     .05       0
  4831.6     .07       0  5452.1     .05       0  8703.9      .1       0
 10477.7     .05       0 11772.5      .1       0 12700.1      .1       0
 14599.2      .1       0 15498.7      .1       0 16695.5     .16       0
 18130.4      .1       0 19154.7      .1       0 21170.3     .16       0
 23387.4      .1       0
Bank Sta=4736.5,5356.8
XS Rating Curve= 0 ,0
Exp/Cntr=0.3,0.1

Type RM Length L Ch R = 1 ,394338  ,1679,1679,1679
BEGIN DESCRIPTION:
PEDERNALES RIVER 158.0
END DESCRIPTION:
XS GIS Cut Line= 3
      2803770.31     10072992.87      2808122.58     10057680.36
       2807665.2      10030937.8
#Sta/Elev= 30
-16424.8 1679.36-15963.5 1661.67  -14343 1632.67-13925.7 1610.55-13358.8 1641.52
-11843.7 1638.72-10233.3 1584.71   -7787  1548.8   -5745 1568.23 -4891.5 1581.93
   -42.8 1517.24  3349.6 1491.16  4821.6 1479.85  4911.6 1463.78  5021.4 1443.79
  5121.7 1465.48  6966.7 1475.61  7974.1 1484.24  9066.8  1493.6 12268.7  1516.5
 14006.5 1528.63 14931.9 1535.09   17000 1564.45 18321.4 1564.27 19263.7  1559.8
 21934.1 1647.54 22212.2 1630.61 22831.4 1672.76 23638.1 1680.72 26240.7 1719.08
#Mann= 19 ,-1 , 0
-16424.8     .16       0-15963.5     .16       0  -14343      .1       0
   -7787      .1       0   -5745      .1       0   -42.8     .05       0
  3349.6      .1       0  4821.6     .07       0  5121.7     .05       0
  6966.7     .05       0  7974.1      .1       0  9066.8      .1       0
 12268.7     .05       0 14006.5      .1       0 14931.9     .05       0
   17000     .05       0 18321.4      .1       0 22212.2     .16       0
 23638.1      .1       0
Bank Sta=4911.6,5121.7
XS Rating Curve= 0 ,0
Exp/Cntr=0.3,0.1

Type RM Length L Ch R = 1 ,392659  ,2353,2353,2353
BEGIN DESCRIPTION:
PEDERNALES RIVER 173.0
END DESCRIPTION:
XS GIS Cut Line= 4
      2807901.95     10071518.02      2809378.08     10052854.51
      2808949.21     10048126.81      2809587.08     10029869.25
#Sta/Elev= 30
-15306.8 1613.52-14665.6 1604.16-11116.6 1584.63 -9659.2 1557.84   -7107 1507.82
 -6159.7 1537.05 -5321.4 1522.59 -3074.4 1558.71 -1019.8 1530.43  3379.6 1489.82
    4701 1471.45  4951.8 1442.95  5453.8  1469.5  5594.7 1449.09  6030.1 1475.73
  7214.3 1471.65  8530.2 1507.39 10568.8 1497.19 11967.4 1510.91 13715.8 1528.76
 14984.2 1541.71 16150.1 1563.96 17945.1  1605.2 19178.6 1611.98 20687.4 1619.43
 21703.4 1683.44 23124.3 1704.94   24033 1681.72 24855.4 1713.53 26430.8 1845.02
#Mann= 20 ,-1 , 0
-15306.8      .1       0-14665.6      .1       0-11116.6     .05       0
 -9659.2      .1       0 -6159.7      .1       0 -1019.8     .05       0
  3379.6     .05       0    4701     .07       0  5453.8     .05       0
  6030.1      .1       0  7214.3      .1       0  8530.2     .05       0
 10568.8      .1       0 11967.4     .05       0 13715.8      .1       0
 14984.2     .05       0 16150.1     .05       0 17945.1      .1       0
 19178.6      .1       0 20687.4      .1       0
Bank Sta=4701,5453.8
XS Rating Curve= 0 ,0
Exp/Cntr=0.3,0.1

Type RM Length L Ch R = 1 ,390306  ,3407,3407,3407
BEGIN DESCRIPTION:
PEDERNALES RIVER 161.0
END DESCRIPTION:
XS GIS Cut Line= 4
      2809582.46     10073323.63      2810418.22     10054496.19
      2811622.25     10033936.43      2810717.27     10029847.03
#Sta/Elev= 30
-18716.8 1665.94-17593.3  1659.3-16406.7 1645.71-13500.6 1586.84-10075.9 1553.76
 -6290.7 1532.89 -5714.1 1482.45 -5529.4 1513.14 -2077.1 1496.38  1136.7 1485.17
  3691.9 1467.24  4494.7 1461.85  4639.4 1461.18  4949.6 1442.12  5050.1 1462.73
  5060.1 1468.97    5208 1474.41  6035.7 1504.86  7006.4 1496.39  8156.2 1502.98
 10401.5 1515.84 14267.6 1537.99   15463 1565.54 17223.8 1605.91 19555.3 1624.54
 20407.1 1623.82 22154.5 1693.73 23074.8 1681.08 24463.7 1772.87 24912.5 1778.15
#Mann= 20 ,-1 , 0
-18716.8      .1       0-17593.3      .1       0-16406.7      .1       0
-13500.6     .16       0-10075.9      .1       0 -5529.4      .1       0
 -2077.1     .05       0  1136.7      .1       0  3691.9      .1       0
  4494.7     .07       0  5060.1      .1       0    5208      .1       0
  7006.4     .05       0  8156.2     .05       0 10401.5      .1       0
 14267.6      .1       0   15463     .05       0 17223.8      .1       0
 19555.3      .1       0 23074.8      .1       0
Bank Sta=4639.4,5050.1
XS Rating Curve= 0 ,0
Exp/Cntr=0.3,0.1

Type RM Length L Ch R = 1 ,386899  ,4143,4143,4143
BEGIN DESCRIPTION:
PEDERNALES RIVER 167.0
END DESCRIPTION:
XS GIS Cut Line= 4
      2810718.33     10072952.21      2811833.35     10054006.53
      2815055.92     10037377.79      2815041.08     10034304.41
#Sta/Elev= 30
-15795.4 1667.01-15212.6 1650.16-14766.6 1638.53-13939.7 1618.39-11108.1 1570.22
 -8894.8  1569.1 -6175.8 1597.86 -4407.2 1528.45 -4063.9 1538.02   -1943 1520.41
 -1380.6 1510.65   580.3 1478.51  1442.9  1467.7  1693.3 1446.86  2127.6 1473.89
  4560.1 1477.02  4765.2 1473.86  4998.8 1436.15  5763.6 1472.35  5894.9 1475.46
  6570.7 1483.53  9466.3 1491.03 10562.2 1486.85 11672.7 1502.31 12471.4 1510.75
 13746.1 1511.84 15898.1 1571.98 18930.1 1621.51 20788.7    1608 23194.6 1688.58
#Mann= 20 ,-1 , 0
-15795.4      .1       0-15212.6      .1       0-14766.6     .05       0
-13939.7      .1       0 -4063.9      .1       0   -1943     .16       0
 -1380.6      .1       0   580.3      .1       0  2127.6     .05       0
  4560.1      .1       0  4765.2     .07       0  5763.6      .1       0
  5894.9      .1       0  6570.7     .05       0  9466.3     .05       0
 10562.2      .1       0 11672.7     .05       0 12471.4      .1       0
 18930.1      .1       0 20788.7      .1       0
Bank Sta=4765.2,5763.6
XS Rating Curve= 0 ,0
Exp/Cntr=0.3,0.1

Type RM Length L Ch R = 1 ,382756  ,5007,5007,5007
BEGIN DESCRIPTION:
PEDERNALES RIVER 169.0
END DESCRIPTION:
XS GIS Cut Line= 4
      2811758.52     10072750.07      2814162.23      10055948.5
      2813875.92     10047804.55      2816029.78     10033351.08
#Sta/Elev= 30
-12492.5 1630.28-12188.8 1625.48-11047.2 1608.52   -9823 1591.49 -8920.2 1582.34
 -8714.2 1599.69 -7066.9 1600.45 -6246.1 1594.29 -4121.2 1616.07 -1582.4 1592.06
  -846.7 1560.74  2189.1 1497.38  3522.8 1485.99  4005.5 1477.35    4695 1469.96
  4724.9 1464.83  4944.9 1432.94  5305.4  1463.7  6518.4 1467.02  7444.6 1469.55
 10583.5 1478.14 12712.8 1480.21 14449.6 1496.98 15524.3  1508.7 17163.3 1537.12
 20828.2 1612.53   22063 1634.94 24009.9  1621.5 24555.5 1637.15 27242.2  1743.2
#Mann= 20 ,-1 , 0
-12492.5      .1       0-12188.8      .1       0-11047.2     .05       0
   -9823      .1       0 -7066.9      .1       0  -846.7      .1       0
  2189.1      .1       0  3522.8      .1       0  4005.5     .05       0
    4695     .07       0  5305.4      .1       0  6518.4      .1       0
  7444.6      .1       0 10583.5     .05       0 12712.8      .1       0
 14449.6     .05       0 15524.3     .05       0 17163.3      .1       0
 20828.2      .1       0 24555.5      .1       0
Bank Sta=4724.9,5305.4
XS Rating Curve= 0 ,0
Exp/Cntr=0.3,0.1

Type RM Length L Ch R = 1 ,377749  ,1142,1142,1142
BEGIN DESCRIPTION:
PEDERNALES RIVER 171.0
END DESCRIPTION:
XS GIS Cut Line= 4
      2812732.11     10072647.22      2815941.29     10054076.34
      2815752.91      10047237.7      2817075.75     10033398.34
#Sta/Elev= 30
  -15837 1644.74-15426.1 1634.03-14930.3 1604.34-14037.7 1612.53-13656.4 1635.02
   -9840 1616.28 -8838.5 1656.94 -7429.9 1655.29 -5269.2 1563.94 -1828.2 1529.25
     927 1507.34  1898.1 1499.54  3104.5 1506.61  3629.5 1487.44 4295.75 1463.48
  5022.2 1424.99  5382.6 1457.11  5422.7 1462.83  6198.3 1467.56  7220.3  1475.4
  8398.7 1484.43 10584.3 1501.99 12382.4 1525.08 13014.3 1537.63 16229.1 1598.02
 17222.8 1593.93 18456.2 1596.03 21835.4 1700.16 22511.8 1687.61 23752.8 1758.16
#Mann= 20 ,-1 , 0
  -15837     .05       0-15426.1      .1       0-14037.7      .1       0
 -7429.9      .1       0 -1828.2     .05       0     927     .05       0
  1898.1      .1       0  3104.5      .1       0  3629.5     .05       0
 4295.75     .07       0  5382.6      .1       0  6198.3     .05       0
  7220.3      .1       0  8398.7      .1       0 10584.3      .1       0
 12382.4      .1       0 13014.3     .05       0 16229.1      .1       0
 17222.8     .05       0 18456.2      .1       0
Bank Sta=4295.75,5422.7
XS Rating Curve= 0 ,0
Exp/Cntr=0.3,0.1

Type RM Length L Ch R = 1 ,376607  ,2218,2218,2218
BEGIN DESCRIPTION:
PEDERNALES RIVER 175.0
END DESCRIPTION:
XS GIS Cut Line= 2
      2816096.61     10072954.17      2817833.24     10033538.01
#Sta/Elev= 30
-15753.4  1726.4-14611.9 1681.52-14125.6 1715.21-13554.4 1759.76-12770.1 1767.22
-10804.1 1663.34-10128.2 1675.52 -7419.4 1622.37 -6834.3 1583.22 -6457.3 1587.41
 -5833.4 1606.45 -4845.7 1568.61 -2420.2 1509.83   -1106 1508.14  3025.2 1490.81
    4622 1458.95  5006.9 1423.05  5308.1 1445.69  6212.9 1463.14 12444.4 1498.31
 14901.9 1549.58 16036.2 1566.78   16887  1577.3 17858.3 1558.34   18681 1579.05
 19733.3  1617.5 21202.4 1657.78 22043.7 1635.65 22674.3  1655.5   23701 1717.11
#Mann= 15 ,-1 , 0
-15753.4     .16       0-14125.6      .1       0-10804.1     .16       0
-10128.2      .1       0 -6457.3      .1       0 -4845.7     .05       0
 -2420.2      .1       0   -1106      .1       0    4622     .07       0
  6212.9      .1       0 14901.9      .1       0 16036.2      .1       0
 17858.3      .1       0   18681      .1       0 19733.3      .1       0
Bank Sta=4622,6212.9
XS Rating Curve= 0 ,0
Exp/Cntr=0.3,0.1

Type RM Length L Ch R = 1 ,374389  ,2360,2360,2360
BEGIN DESCRIPTION:
PEDERNALES RIVER 177.0
END DESCRIPTION:
XS GIS Cut Line= 3
      2817292.23     10072676.26      2819738.83      10043279.4
      2826480.51     10031645.27
#Sta/Elev= 30
-15577.2 1723.55-14611.3 1735.46-13989.2 1858.65-13788.6 1870.84-13633.1 1859.56
-13271.6 1758.16-12867.1 1730.55-10438.2 1727.98 -7450.2 1589.45 -4630.2 1545.66
 -3314.7 1525.23  -619.1 1483.37   344.1 1490.49  3161.6 1477.59  4624.9 1455.63
    5016 1422.35  5299.2 1450.76  5929.9 1464.83 10048.3 1478.72 11011.6 1490.78
 13378.2 1504.85 14520.8 1522.12 17052.5 1538.64 20064.9 1612.01 21713.4 1617.02
 22224.1 1653.67 23626.3 1642.59 25163.6 1699.12 26035.8 1665.01 27367.6 1729.87
#Mann= 20 ,-1 , 0
-15577.2      .1       0-13788.6      .1       0-12867.1      .1       0
-10438.2      .1       0 -7450.2     .05       0 -4630.2     .05       0
 -3314.7     .05       0  -619.1     .05       0   344.1      .1       0
  3161.6      .1       0  4624.9     .07       0  5299.2      .1       0
  5929.9      .1       0 10048.3      .1       0 11011.6      .1       0
 13378.2     .05       0 14520.8     .05       0 17052.5      .1       0
 21713.4      .1       0 23626.3      .1       0
Bank Sta=4624.9,5299.2
XS Rating Curve= 0 ,0
Exp/Cntr=0.3,0.1

Type RM Length L Ch R = 1 ,372029  ,1781,1781,1781
BEGIN DESCRIPTION:
PEDERNALES RIVER 179.0
END DESCRIPTION:
XS GIS Cut Line= 4
      2817959.75      10072809.1      2820180.08      10055257.2
      2822256.75      10045082.1      2827177.43     10032148.46
#Sta/Elev= 30
-14020.6 1712.35-13881.5 1705.43-12890.3 1712.63  -10644 1663.47 -9451.6 1694.25
 -8018.9 1684.47 -5736.9 1600.72   -3199 1528.75 -1917.2 1507.52   767.9 1500.95
  4638.7 1456.29  4739.8 1454.26  4980.9 1422.37  5379.1 1442.77  5399.6 1450.11
  7445.6 1469.32  9337.8 1495.13 11083.3 1518.94 13008.5 1545.21 14970.1 1571.81
   15745 1582.24 16897.5 1602.33 17847.2 1631.31 19413.7 1635.46 20307.1 1692.62
 22901.3 1644.35   24815 1710.88   25525 1769.94 27178.4 1720.12 27894.1 1774.06
#Mann= 19 ,-1 , 0
-14020.6     .16       0-13881.5      .1       0-12890.3      .1       0
 -9451.6      .1       0 -5736.9     .05       0   -3199      .1       0
 -1917.2     .05       0   767.9      .1       0  4638.7     .07       0
  5379.1      .1       0  7445.6     .05       0  9337.8      .1       0
 11083.3     .05       0 13008.5      .1       0 14970.1     .05       0
   15745      .1       0 16897.5     .05       0 17847.2      .1       0
 20307.1      .1       0
Bank Sta=4739.8,5399.6
XS Rating Curve= 0 ,0
Exp/Cntr=0.3,0.1

Type RM Length L Ch R = 1 ,370248  ,1734,1734,1734
BEGIN DESCRIPTION:
PEDERNALES RIVER 182.0
END DESCRIPTION:
XS GIS Cut Line= 4
      2819657.08     10073550.56      2821379.34     10056806.47
       2824536.4     10047024.31      2827859.34      10032523.6
#Sta/Elev= 30
-14395.4 1723.61  -12537 1647.41-10819.8 1619.95 -9645.2 1658.73   -7886 1644.57
 -6607.3 1591.81   -5679 1578.76 -4104.4 1531.11 -2994.8 1494.55   915.2 1485.95
  4751.6 1444.09  4972.1 1422.44  5245.4 1443.88  5314.7 1446.55  6975.1 1452.97
  9420.2  1501.8 11886.5 1507.25 14040.2 1521.28 15376.3 1540.61 17430.7 1588.01
 18338.7 1608.96 19601.5 1674.76 21467.7 1618.52 21884.7 1644.46 23177.4 1692.55
 23808.8  1679.8   25281 1756.44 26089.2 1716.18 26897.4 1712.29 27592.6 1756.49
#Mann= 11 ,-1 , 0
-14395.4      .1       0  -12537      .1       0   -5679      .1       0
 -4104.4      .1       0  4751.6     .07       0  5314.7      .1       0
 11886.5      .1       0 14040.2     .05       0 15376.3      .1       0
 17430.7      .1       0 21884.7      .1       0
Bank Sta=4751.6,5245.4
XS Rating Curve= 0 ,0
Exp/Cntr=0.3,0.1

Type RM Length L Ch R = 1 ,368514  ,2394,2394,2394
BEGIN DESCRIPTION:
PEDERNALES RIVER 183.0
END DESCRIPTION:
XS GIS Cut Line= 4
      2820931.04     10072473.22      2822942.77     10056915.43
      2826031.04     10049226.76      2828201.57     10034887.24
#Sta/Elev= 30
-12529.7  1681.3-11597.4 1645.64-11105.3 1649.98 -9434.7 1597.86 -8541.5  1602.2
 -7770.9 1594.53 -7289.1 1615.85 -2236.6 1510.15  -464.9 1494.94   414.6 1475.73
  1233.4 1450.74  1756.1 1468.51    4579  1445.4  4603.2 1443.31    4931 1422.96
 5288.87 1444.64  8558.1 1462.01 10761.8 1480.89 11183.8 1477.88 12773.7 1492.96
 14651.6    1527 15381.8 1535.79 15834.1 1541.22 17786.8  1580.4 18515.1 1598.68
 19474.7 1617.78 21408.6 1582.99 22681.4 1668.96 24085.9  1633.2 25946.2  1723.8
#Mann= 17 ,-1 , 0
-12529.7      .1       0-11597.4      .1       0 -8541.5      .1       0
 -2236.6     .05       0  -464.9     .05       0   414.6      .1       0
    4579     .07       0 5288.87      .1       0  8558.1      .1       0
 10761.8     .16       0 11183.8      .1       0 12773.7     .05       0
 14651.6      .1       0 15381.8     .05       0 15834.1      .1       0
 17786.8     .16       0 18515.1      .1       0
Bank Sta=4603.2,5288.87
XS Rating Curve= 0 ,0
Exp/Cntr=0.3,0.1

Type RM Length L Ch R = 1 ,366120  ,2358,2358,2358
BEGIN DESCRIPTION:
PEDERNALES RIVER 184.0
END DESCRIPTION:
XS GIS Cut Line= 4
      2822971.87     10071697.04      2825251.45     10058215.02
      2826478.24      10051013.8        2829052.     10035637.37
#Sta/Elev= 30
-10691.2 1715.32-10467.8 1706.61 -6186.4 1554.71 -5108.4 1552.65 -2029.5 1540.53
 -1002.8 1533.61   292.9 1512.45   988.6 1520.57  4058.8 1487.56  4667.4 1445.84
    4717 1442.44  5022.9 1414.83  5379.3 1443.56  6683.5 1448.32  7142.6 1429.47
  7817.3 1447.79  8058.1  1436.1  9449.1 1451.04 11250.2 1473.33 13399.5 1506.01
   15084 1510.24 16060.6 1523.25 17870.8 1554.82 19241.7 1563.61 19957.3 1575.54
 21301.2 1571.85   22674 1637.09 23569.5 1598.31 25157.9 1714.17 25877.5 1732.75
#Mann= 17 ,-1 , 0
-10691.2     .05       0-10467.8      .1       0 -5108.4     .05       0
 -2029.5      .1       0 -1002.8      .1       0   988.6      .1       0
  4667.4     .07       0  5379.3      .1       0  9449.1      .1       0
 11250.2      .1       0 13399.5     .05       0   15084      .1       0
 16060.6     .05       0 17870.8      .1       0 19241.7      .1       0
 19957.3      .1       0 21301.2      .1       0
Bank Sta=4717,5379.3
XS Rating Curve= 0 ,0
Exp/Cntr=0.3,0.1

Type RM Length L Ch R = 1 ,363762  ,1481,1481,1481
BEGIN DESCRIPTION:
PEDERNALES RIVER 185.0
END DESCRIPTION:
XS GIS Cut Line= 4
       2826509.8     10070763.35      2827973.74     10057434.22
      2827105.52     10052974.65      2829645.04      10035968.7
#Sta/Elev= 30
-11015.5 1659.43 -9229.9 1636.21   -8028  1586.9 -7591.6 1597.13 -5073.2 1543.45
 -3509.1  1517.2 -2823.2 1506.61   189.5 1494.01  4482.8 1435.99  4488.1 1435.24
  4962.8  1410.8    5257 1434.44  5572.9 1421.34  6847.3 1466.83  8767.3 1483.64
  9738.9 1488.86 10717.8    1503 11534.1 1491.89 12351.5 1488.47 13567.2 1495.96
 14538.4 1510.78 16235.3 1528.82 18637.5  1548.8 19172.2 1545.79 20587.7 1599.15
 21467.4 1578.67 22539.1 1660.31 22900.1 1668.01 23337.9 1715.16 24131.6 1704.24
#Mann= 16 ,-1 , 0
-11015.5      .1       0 -9229.9      .1       0 -5073.2      .1       0
 -3509.1     .05       0 -2823.2      .1       0  4482.8     .07       0
    5257      .1       0  8767.3      .1       0  9738.9      .1       0
 10717.8     .05       0 11534.1      .1       0 12351.5     .05       0
 13567.2     .05       0 14538.4     .05       0 16235.3      .1       0
 18637.5      .1       0
Bank Sta=4488.1,5257
XS Rating Curve= 0 ,0
Exp/Cntr=0.3,0.1

Type RM Length L Ch R = 1 ,362281  ,1580,1580,1580
BEGIN DESCRIPTION:
PEDERNALES RIVER 195.0
END DESCRIPTION:
XS GIS Cut Line= 4
       2828373.3     10069212.63      2829016.97     10056416.02
      2828368.38     10051742.08      2830128.02     10036408.63
#Sta/Elev= 30
  -10069 1646.51 -8273.5 1627.93 -7479.9 1600.03 -6481.6 1600.54 -5612.3  1563.6
   -3359 1509.26 -2899.3 1503.75    1531 1456.24  1684.7 1474.05  3789.4 1434.95
  4588.4 1432.78  4603.7 1430.14  4997.2 1409.61  5310.4 1430.77  6390.8 1457.48
    7822 1481.77    9323 1466.48 10050.3  1473.7 10742.2 1470.69 12094.1 1493.86
 13781.2 1503.67 15840.3 1514.41 16239.6 1518.96 17817.4  1539.1 18560.6 1544.74
 19138.4 1550.08 20027.8 1567.29 20515.6 1588.93 21712.6 1652.45 22896.6  1687.1
#Mann= 19 ,-1 , 0
  -10069      .1       0 -5612.3      .1       0   -3359      .1       0
 -2899.3      .1       0    1531      .1       0  4588.4     .07       0
  5310.4      .1       0  6390.8      .1       0    7822      .1       0
 10050.3      .1       0 12094.1     .05       0 13781.2     .05       0
 15840.3     .16       0 16239.6      .1       0 17817.4      .1       0
 18560.6     .16       0 19138.4      .1       0 20027.8     .16       0
 20515.6      .1       0
Bank Sta=4603.7,5310.4
XS Rating Curve= 0 ,0
Exp/Cntr=0.3,0.1

Type RM Length L Ch R = 1 ,360701  ,1418,1418,1418
BEGIN DESCRIPTION:
PEDERNALES RIVER 197.0
END DESCRIPTION:
XS GIS Cut Line= 3
      2829409.28     10068791.11        2830219.     10055725.28
      2830652.37     10036480.06
#Sta/Elev= 30
 -9325.6 1637.23 -8562.6 1603.84 -6991.6 1578.92 -5864.7  1602.3 -5023.5 1590.12
   -4520 1575.06   -3788 1547.73 -1902.7 1507.86     117 1491.47  2219.8 1441.05
  2863.8 1459.57  4607.1 1435.64  5026.9 1407.09  5497.3 1434.61  6775.7 1440.71
  8271.5 1441.34  8945.1 1451.28  9674.9 1469.72 11304.1 1492.44 11923.9 1503.67
 14626.6 1520.89   16310  1533.7 16771.4 1547.41   18031 1578.81 18623.9  1601.8
   20201 1611.98 20691.1 1594.48 20851.2 1609.83 22176.2 1621.73 23015.4 1665.33
#Mann= 17 ,-1 , 0
 -9325.6      .1       0 -8562.6      .1       0 -5023.5     .16       0
   -4520      .1       0   -3788     .05       0 -1902.7      .1       0
  4607.1     .07       0  6775.7      .1       0  8271.5     .16       0
  8945.1     .05       0  9674.9      .1       0 11304.1     .05       0
 11923.9      .1       0 14626.6      .1       0   16310      .1       0
 16771.4      .1       0   18031      .1       0
Bank Sta=4607.1,5497.3
XS Rating Curve= 0 ,0
Exp/Cntr=0.3,0.1

Type RM Length L Ch R = 1 ,359283  ,1624,1624,1624
BEGIN DESCRIPTION:
PEDERNALES RIVER 198.0
END DESCRIPTION:
XS GIS Cut Line= 2
      2830838.18     10068359.27      2832736.19     10036453.37
#Sta/Elev= 30
 -8888.9 1626.17 -8492.7 1606.82 -7818.9 1601.01 -7204.7 1584.79 -6256.3 1541.33
 -5765.8 1538.96 -5029.8  1563.6 -3840.1 1538.87   -3033 1510.62 -1823.5 1503.93
  3090.3 1432.74  4640.5 1428.43  5020.9 1406.56  5301.7 1426.05  5381.8 1426.91
  6784.3 1418.62  7413.7 1435.87    9458 1483.48 10972.5 1499.97 12254.3 1528.59
 14037.9 1544.83 15021.2 1568.85 18031.8 1615.12 19208.1 1640.62 20163.8 1688.12
 20852.4 1695.53 21590.4  1664.1 21852.3 1670.57 22401.9 1653.77 23073.4 1663.07
#Mann= 19 ,-1 , 0
 -8888.9      .1       0 -7818.9      .1       0 -7204.7     .16       0
 -6256.3      .1       0 -5029.8     .16       0 -3840.1     .05       0
 -1823.5      .1       0  3090.3      .1       0  4640.5     .07       0
  5381.8      .1       0  7413.7     .05       0    9458      .1       0
 10972.5     .05       0 12254.3      .1       0 14037.9     .16       0
 15021.2      .1       0 18031.8      .1       0 19208.1      .1       0
 20852.4      .1       0
Bank Sta=4640.5,5301.7
XS Rating Curve= 0 ,0
Exp/Cntr=0.3,0.1

Type RM Length L Ch R = 1 ,357659  ,1684,1684,1684
BEGIN DESCRIPTION:
PEDERNALES RIVER 202.0
END DESCRIPTION:
XS GIS Cut Line= 2
      2832084.25     10068686.92      2834362.54     10041213.02
#Sta/Elev= 30
 -8990.4 1625.99 -8638.9 1595.97 -8017.7 1570.58 -7306.1  1550.5 -5958.3 1536.33
 -5431.7 1523.79 -4241.3 1517.37 -2760.5  1492.1 -1491.7 1476.71   876.5 1464.72
  2742.9 1428.81  4639.4  1424.4  4849.9  1406.6  5271.6 1413.09  5351.8 1424.38
    5392  1424.7  6613.6 1432.59  8033.6 1438.85  8935.3 1446.15 11804.8 1496.13
 12275.5 1474.15 12886.6 1497.38 13752.2  1517.6 14165.9 1513.43 14733.9 1537.33
 16218.6 1561.22   16801 1586.08 17169.4  1584.5 18296.4 1649.89 18577.8 1653.51
#Mann= 18 ,-1 , 0
 -8990.4      .1       0 -8017.7      .1       0 -5958.3     .05       0
 -5431.7      .1       0 -4241.3     .05       0 -2760.5      .1       0
 -1491.7      .1       0  4639.4     .07       0    5392      .1       0
  6613.6      .1       0  8033.6     .05       0  8935.3      .1       0
 11804.8     .16       0 12886.6      .1       0 14165.9      .1       0
 16218.6      .1       0 17169.4      .1       0 18296.4      .1       0
Bank Sta=4639.4,5351.8
XS Rating Curve= 0 ,0
Exp/Cntr=0.3,0.1

Type RM Length L Ch R = 1 ,355975  ,2218,2218,2218
BEGIN DESCRIPTION:
PEDERNALES RIVER 204.0
END DESCRIPTION:
XS GIS Cut Line= 3
      2833517.66     10068394.58      2834704.87     10056693.43
      2835878.53     10041581.77
#Sta/Elev= 30
 -8174.4 1624.62 -7409.6  1601.2 -6568.4 1608.53 -6131.8 1602.12 -5343.6 1562.32
 -4749.8 1552.79 -4283.7 1562.63 -3368.7 1538.26 -2448.9 1525.78 -1620.6 1498.21
 -1028.8 1491.67  -192.2 1480.16  1655.7  1476.8  4509.3 1426.31  4900.2 1397.64
  5241.5  1421.6  6386.1  1431.9  7426.3 1424.45  8782.1  1426.4  9379.6 1450.29
 10927.8 1459.58 12244.4  1476.4 12996.2 1497.46   13838 1507.66 14550.2 1513.07
 15280.1 1541.05 16092.4 1579.12 16459.8 1582.22 17130.5 1578.29   18744 1656.34
#Mann= 18 ,-1 , 0
 -8174.4      .1       0 -6568.4      .1       0 -3368.7      .1       0
 -2448.9     .05       0 -1620.6      .1       0 -1028.8     .05       0
  -192.2      .1       0  1655.7      .1       0  4509.3     .07       0
  5241.5      .1       0  6386.1      .1       0  7426.3     .05       0
 10927.8     .05       0 12244.4      .1       0 12996.2     .05       0
   13838      .1       0 15280.1      .1       0 16459.8     .05       0
Bank Sta=4509.3,5241.5
XS Rating Curve= 0 ,0
Exp/Cntr=0.3,0.1

Type RM Length L Ch R = 1 ,353757  ,1662,1662,1662
BEGIN DESCRIPTION:
PEDERNALES RIVER 208.0
END DESCRIPTION:
XS GIS Cut Line= 3
      2835258.77     10069955.71      2836903.99     10056775.16
      2837032.78     10041650.74
#Sta/Elev= 30
-10353.8 1577.75 -9670.8 1548.96 -8783.3 1550.04 -8068.1 1531.98 -6159.5 1512.52
 -5556.4  1520.1   -4346 1520.09 -4065.6 1507.51 -3710.7 1491.98 -3261.2 1499.78
 -2646.7 1520.59 -2001.3 1521.46 -1517.2 1504.02  -878.9 1519.86   661.1 1475.97
  4570.5  1421.6  4890.5 1399.34  5270.5 1411.43  5570.3 1396.95  6095.6 1419.21
  6180.6 1424.44  6620.2 1434.75  7887.1  1457.6  8982.5 1479.78   11500 1510.36
 12189.5 1513.41 14860.9 1569.25 15970.9 1556.12 17973.2 1645.27   18054 1648.06
#Mann= 14 ,-1 , 0
-10353.8      .1       0 -8068.1      .1       0 -5556.4      .1       0
 -4065.6      .1       0 -3261.2      .1       0 -2646.7      .1       0
  4570.5     .07       0  6180.6     .16       0  6620.2      .1       0
  7887.1      .1       0  8982.5     .05       0   11500      .1       0
 12189.5      .1       0 17973.2     .05       0
Bank Sta=4570.5,6095.6
XS Rating Curve= 0 ,0
Exp/Cntr=0.3,0.1

Type RM Length L Ch R = 1 ,352095  ,1902,1902,1902
BEGIN DESCRIPTION:
PEDERNALES RIVER 210.0
END DESCRIPTION:
XS GIS Cut Line= 2
      2837787.14     10070096.44      2838987.24     10043764.67
#Sta/Elev= 30
-10881.4 1592.05-10328.1 1554.19 -9436.1 1545.25 -8307.3  1543.2 -7221.9 1521.48
   -6311 1506.76   -5106 1491.63 -4240.2 1474.79 -3240.8 1456.54 -1516.7 1472.44
 -1080.9 1478.85  -127.5  1454.9  2114.8 1435.84  2184.9 1421.23    2365 1434.57
  4487.2 1410.93  4537.3 1408.51  4927.4 1392.53    5228 1411.47    5238 1411.67
  6649.5 1426.32  6899.7 1448.35  7890.8 1478.56  9135.7 1494.97   10376 1503.45
 11674.7 1497.18 13707.2 1582.19 14948.1 1624.48 15422.7 1621.44 15477.7 1618.63
#Mann= 14 ,-1 , 0
-10881.4      .1       0 -9436.1      .1       0 -8307.3      .1       0
 -7221.9     .05       0   -6311      .1       0   -5106     .05       0
 -4240.2      .1       0 -1516.7      .1       0  4537.3     .07       0
    5238      .1       0  9135.7     .05       0   10376      .1       0
 13707.2      .1       0 15422.7     .16       0
Bank Sta=4487.2,5228
XS Rating Curve= 0 ,0
Exp/Cntr=0.3,0.1

Type RM Length L Ch R = 1 ,350193  ,2346,2346,2346
BEGIN DESCRIPTION:
PEDERNALES RIVER 212.0
END DESCRIPTION:
XS GIS Cut Line= 4
      2839402.01     10068466.09      2840093.69     10056813.93
      2841262.29     10046652.52      2840370.16     10043121.44
#Sta/Elev= 30
 -9207.8 1613.97 -8604.4 1602.25 -7794.2 1569.15 -6335.1  1525.6 -4244.9 1482.93
 -3921.8 1476.77 -3229.7  1466.9 -1272.3 1441.39  -800.7 1431.44   -72.3 1459.82
    1793 1429.06    3337 1407.81  4377.6 1406.71  4397.7 1407.19    4931 1392.57
    5172 1405.51  5565.4 1404.22  6978.2  1441.7  7368.3 1453.85  8102.6 1449.96
  8533.5  1457.1  8854.2  1464.2 10457.4 1497.77 11975.6 1513.04 13590.1 1518.94
 14154.8 1515.96 15098.7 1550.76   15545 1548.75 16330.9 1590.63 16335.3  1590.8
#Mann= 17 ,-1 , 0
 -9207.8      .1       0 -7794.2      .1       0 -6335.1      .1       0
 -4244.9      .1       0 -3921.8     .05       0 -3229.7      .1       0
 -1272.3      .1       0    1793      .1       0  4377.6     .07       0
    5172      .1       0  6978.2     .16       0  8102.6      .1       0
  8533.5     .05       0  8854.2      .1       0 11975.6     .05       0
 13590.1      .1       0 16330.9      .1       0
Bank Sta=4397.7,5172
XS Rating Curve= 0 ,0
Exp/Cntr=0.3,0.1

Type RM Length L Ch R = 1 ,347847  ,2460,2460,2460
BEGIN DESCRIPTION:
PEDERNALES RIVER 214.0
END DESCRIPTION:
XS GIS Cut Line= 4
      2840990.82     10068980.41      2841513.52     10057656.23
      2842807.67     10050741.57      2841417.08     10042969.15
#Sta/Elev= 30
 -7927.4 1595.57 -7289.1 1562.28 -6739.5 1542.61 -6035.3 1538.47 -5208.9 1519.41
 -4619.5 1503.47 -3437.9 1501.16 -2675.1 1502.96 -2141.6 1486.23 -1147.7 1467.21
    -492 1471.06   772.3  1436.8  1761.9 1424.52  2716.7 1418.72    4553 1400.47
  4988.9 1381.88  5547.8 1397.52  5568.2 1402.93  6163.9 1409.65  7165.4 1444.77
  7277.4 1432.05  8244.7 1467.07   10636 1502.21 11987.7 1502.69 13890.2 1504.44
 14835.4 1501.89 15575.8 1502.42 16136.8 1490.92 18265.9 1533.21 18339.4 1532.48
#Mann= 20 ,-1 , 0
 -7927.4      .1       0 -7289.1      .1       0 -6035.3     .05       0
 -5208.9      .1       0 -3437.9     .05       0 -2141.6      .1       0
   772.3      .1       0  1761.9      .1       0  2716.7      .1       0
    4553     .07       0  5547.8      .1       0  6163.9      .1       0
  8244.7      .1       0   10636     .05       0 11987.7      .1       0
 13890.2     .05       0 14835.4      .1       0 15575.8     .05       0
 16136.8      .1       0 18265.9     .05       0
Bank Sta=4553,5568.2
XS Rating Curve= 0 ,0
Exp/Cntr=0.3,0.1

Type RM Length L Ch R = 1 ,345387  ,2290,2290,2290
BEGIN DESCRIPTION:
PEDERNALES RIVER 218.0
END DESCRIPTION:
XS GIS Cut Line= 3
      2842265.04     10068225.88      2844997.45     10051593.26
      2841237.13     10041844.08
#Sta/Elev= 30
 -6639.7 1588.19   -5961 1570.15   -4809 1567.25 -4119.7 1565.52 -2502.8 1513.77
 -2272.2 1518.78 -1187.7  1496.3  -700.5 1486.48   935.8 1453.49  2679.9 1419.77
  3509.2  1412.4  4454.3 1402.38    4638 1392.68  4965.7 1373.38  5410.4 1389.14
  7369.4 1438.42  8161.2 1454.14  8735.8 1463.08  9713.1 1470.86   10835 1472.66
 11361.5 1485.96 14475.9 1481.11 15063.7 1488.78 15644.8 1476.57 16459.3  1484.9
 17502.9 1479.07 17854.4 1487.66 18577.3  1505.7 19691.9 1523.92 20665.1 1532.46
#Mann= 20 ,-1 , 0
 -6639.7      .1       0   -5961     .05       0   -4809      .1       0
 -1187.7      .1       0  -700.5      .1       0   935.8      .1       0
  2679.9     .05       0  3509.2      .1       0    4638     .07       0
  5410.4     .05       0  5410.4      .1       0  7369.4      .1       0
  8161.2      .1       0  8735.8     .05       0  9713.1     .05       0
 14475.9     .16       0 16459.3     .05       0 17854.4      .1       0
 18577.3      .1       0 19691.9     .05       0
Bank Sta=4638,5410.4
XS Rating Curve= 0 ,0
Exp/Cntr=0.3,0.1

Type RM Length L Ch R = 1 ,343097  ,2380,2380,2380
BEGIN DESCRIPTION:
PEDERNALES RIVER 221.0
END DESCRIPTION:
XS GIS Cut Line= 4
      2843044.93     10068084.66      2845634.17     10060754.77
      2847633.18      10050570.2      2846027.55     10039857.12
#Sta/Elev= 30
 -5941.9 1539.43 -5491.4 1527.92 -4197.6 1522.42 -2792.9 1488.81   -1652 1455.12
  -215.5 1481.81   637.7 1472.61  1834.9 1461.23  2800.2 1432.72  3920.6 1407.24
  4778.1 1387.74    4996 1366.64  5356.3 1389.86  6017.4 1393.36  6710.3 1397.03
  7771.8 1402.46  9032.4 1406.04 11008.8 1411.65 14723.5  1420.7 16597.5 1421.27
 16661.5 1433.29 16730.7 1419.34 17199.4 1461.21   17805 1461.72 19010.6    1479
 20652.2 1518.98   21486 1554.29 21990.9 1571.33 22912.5 1574.94 23043.5 1573.94
#Mann= 20 ,-1 , 0
 -5941.9      .1       0 -5491.4      .1       0 -4197.6     .05       0
 -2792.9      .1       0   637.7      .1       0  2800.2      .1       0
  3920.6      .1       0  4778.1     .07       0  5356.3      .1       0
  6017.4      .1       0  6710.3      .1       0  7771.8      .1       0
  9032.4      .1       0 11008.8     .05       0 14723.5      .1       0
   17805      .1       0 19010.6      .1       0 20652.2      .1       0
   21486     .16       0 22912.5     .16       0
Bank Sta=4778.1,5356.3
XS Rating Curve= 0 ,0
Exp/Cntr=0.3,0.1

Type RM Length L Ch R = 1 ,340717  ,2338,2338,2338
BEGIN DESCRIPTION:
PEDERNALES RIVER 225.0
END DESCRIPTION:
XS GIS Cut Line= 3
      2847355.22     10073415.11      2848828.15     10055098.89
       2849098.7     10038573.25
#Sta/Elev= 30
-10784.6 1576.44 -9464.6 1520.25 -8696.5 1488.64 -7418.4 1503.51 -5335.7 1409.02
 -5141.1 1420.65 -3850.9 1384.61 -3322.7 1435.49 -2250.8 1433.56 -1576.7 1435.07
    -781 1400.77   542.2 1443.15  1292.6  1432.6  4566.2 1389.04  5017.4 1366.58
  5412.7 1386.56    5439  1387.8  8914.1 1395.21  9872.7 1400.88 10399.9 1421.35
 10906.3 1396.04   12160 1407.93 13088.8 1418.47 13412.7 1401.15 14023.2 1439.99
 15742.1 1472.85 19124.8 1480.47 20367.6 1520.13 21268.2 1499.71 24118.6 1599.65
#Mann= 16 ,-1 , 0
-10784.6      .1       0 -9464.6      .1       0 -7418.4      .1       0
 -5141.1      .1       0 -2250.8      .1       0  1292.6      .1       0
  4566.2     .07       0  5412.7      .1       0  8914.1     .05       0
  9872.7     .16       0 10399.9      .1       0   12160      .1       0
 13088.8      .1       0 15742.1      .1       0 19124.8      .1       0
 21268.2      .1       0
#XS Ineff= 2 , 0
          590.91 1445.4310409.09         1422.59
Permanent Ineff=
       F       F
Bank Sta=4566.2,5439
XS Rating Curve= 0 ,0
Exp/Cntr=0.3,0.1

Type RM Length L Ch R = 1 ,338379  ,3023,3023,3023
BEGIN DESCRIPTION:
PEDERNALES RIVER 234.0
END DESCRIPTION:
XS GIS Cut Line= 3
      2849717.75     10073304.95       2849366.9     10062189.14
      2854406.54     10047528.08
#Sta/Elev= 30
 -9440.3 1596.96 -9329.7 1593.21 -8905.5 1574.67 -8173.3 1552.06 -6587.7 1508.75
 -4816.8 1422.24 -4064.2 1416.63 -3844.8 1416.69 -3281.5 1429.52 -1979.5 1381.35
 -1535.1 1362.51 -1465.1 1393.54   -1315  1403.5  -405.4 1387.64     786 1382.02
    1681 1407.26  3780.5  1380.7  4520.7 1374.43  4541.8 1369.86    4880 1361.96
  5430.1 1374.15  6527.7 1390.17  8308.6 1409.35 13269.4 1524.84 14097.1 1597.13
 14450.1 1579.45 15692.9 1540.71 16277.9 1543.98 16534.3 1553.28 17184.1 1590.02
#Mann= 17 ,-1 , 0
 -9440.3      .1       0 -9329.7     .16       0 -8905.5      .1       0
 -8173.3      .1       0 -4064.2     .05       0 -3844.8      .1       0
 -1979.5      .1       0  -405.4      .1       0  3780.5     .16       0
  4541.8     .07       0  5430.1     .16       0  6527.7      .1       0
  8308.6      .1       0 14450.1      .1       0 15692.9     .16       0
 16277.9     .05       0 16534.3      .1       0
#XS Ineff= 2 , 0
        -1238.64 1405.38
Permanent Ineff=
       F       F
Bank Sta=4520.7,5430.1
XS Rating Curve= 0 ,0
Exp/Cntr=0.3,0.1

Type RM Length L Ch R = 1 ,335356  ,4395,4395,4395
BEGIN DESCRIPTION:
PEDERNALES RIVER 236.0
END DESCRIPTION:
XS GIS Cut Line= 3
      2850550.14     10073384.54      2850737.05     10063733.67
      2856145.26      10047340.3
#Sta/Elev= 30
 -6568.9 1567.18 -4242.1 1505.52  1505.1 1375.76  2263.6 1339.65  2499.4 1353.22
  2901.2 1360.89  3073.7 1364.19  3252.2 1348.63  3710.5  1362.8  4160.3 1351.12
  4186.8 1350.87  4318.8 1337.63  5335.2 1351.76  5851.8 1360.72  6598.2 1374.33
  7034.5 1382.41  8785.8 1412.53  9611.4 1406.36  9864.8 1416.41   11263 1459.11
 12697.7 1423.75 12950.4 1432.36 13408.2 1441.44 14037.7 1461.25 15523.5 1474.38
 16366.9 1492.49   18027 1530.86   18625 1546.93 19095.2 1562.58 20346.2 1634.14
#Mann= 19 ,-1 , 0
 -6568.9      .1       0 -4242.1      .1       0  1505.1      .1       0
  2499.4     .16       0  2901.2      .1       0  4160.3     .07       0
  5335.2      .1       0  5851.8      .1       0  6598.2     .16       0
  7034.5      .1       0  9864.8      .1       0   11263      .1       0
 12950.4      .1       0 13408.2     .05       0 14037.7      .1       0
 15523.5      .1       0 16366.9      .1       0   18027     .16       0
   18625      .1       0
Bank Sta=4186.8,5335.2
XS Rating Curve= 0 ,0
Exp/Cntr=0.3,0.1

Type RM Length L Ch R = 1 ,330961  ,2429,2429,2429
BEGIN DESCRIPTION:
PEDERNALES RIVER 245.0
END DESCRIPTION:
XS GIS Cut Line= 2
      2851387.65     10075004.99       2856903.7     10049735.63
#Sta/Elev= 30
 -5133.1 1594.45 -4820.9  1578.3 -3361.4 1501.28 -2756.7 1474.66 -1955.5 1476.02
  -714.5 1457.01   585.9 1422.19  1245.8 1415.06  3404.6 1353.42  3629.8 1337.33
  3762.2 1345.37  4407.6 1357.18  4598.6 1337.31  4833.3 1311.11  5052.5 1312.79
  5124.1 1328.69  5161.5 1336.24  5286.1 1341.86  5866.2 1363.44  6865.2 1373.99
  9956.4 1408.72 10644.1 1416.45 11879.8 1430.33 13097.6 1441.95 14056.8 1466.93
 15780.7 1474.69 17851.6 1490.07 19579.6 1576.03 20519.9 1609.28 20731.3 1599.49
#Mann= 20 ,-1 , 0
 -5133.1     .16       0 -4820.9      .1       0 -3361.4     .05       0
 -1955.5      .1       0  -714.5      .1       0   585.9      .1       0
  1245.8      .1       0  3762.2      .1       0  4598.6     .07       0
  5124.1      .1       0  5286.1      .1       0  6865.2      .1       0
  9956.4      .1       0 10644.1      .1       0 11879.8      .1       0
 14056.8      .1       0 15780.7      .1       0 17851.6      .1       0
 19579.6     .16       0 20519.9     .16       0
Bank Sta=4598.6,5161.5
XS Rating Curve= 0 ,0
Exp/Cntr=0.3,0.1

Type RM Length L Ch R = 1 ,328532  ,3234,3234,3234
BEGIN DESCRIPTION:
PEDERNALES RIVER 246.0
END DESCRIPTION:
XS GIS Cut Line= 3
      2851978.42     10075500.48       2857915.6     10060218.48
      2857980.31      10050453.1
#Sta/Elev= 30
 -4639.8 1582.08 -3631.6    1540 -1431.8 1452.57  -531.1 1442.98   533.1 1443.61
    1224 1419.65  1658.9 1424.14  4690.2 1332.96    4707 1329.68  4766.8  1326.5
  4797.5 1312.59  5038.7 1302.17  5400.8 1328.75  5419.7 1328.54  6649.5 1374.32
  7085.2 1400.56  7616.8 1402.42  8984.5 1430.16 10122.1 1446.97 10819.3 1438.96
   11420 1439.16 12164.2 1457.93 13012.9 1473.67 14026.5 1492.47 14735.1 1505.09
 18329.9 1551.96 19374.2 1554.04 20199.9 1540.81 21086.6 1607.43 21520.6  1616.8
#Mann= 19 ,-1 , 0
 -4639.8      .1       0 -3631.6      .1       0 -1431.8     .16       0
  -531.1     .16       0  1658.9      .1       0  4690.2     .07       0
  5419.7     .16       0  6649.5      .1       0  7616.8      .1       0
  8984.5     .16       0 10122.1      .1       0 10819.3     .16       0
 12164.2      .1       0 13012.9     .05       0 14026.5      .1       0
 14735.1      .1       0 18329.9     .16       0 19374.2     .16       0
 21086.6     .16       0
Bank Sta=4707,5400.8
XS Rating Curve= 0 ,0
Exp/Cntr=0.3,0.1

Type RM Length L Ch R = 1 ,319801  ,2059,2059,2059
BEGIN DESCRIPTION:
PEDERNALES RIVER 254.0
END DESCRIPTION:
XS GIS Cut Line= 4
       2854683.8     10078565.79      2863621.89     10070807.71
      2864440.18     10057090.95      2860494.53     10051400.15
#Sta/Elev= 30
-10970.2 1560.56-10562.2 1543.46 -8470.4 1471.26   -4927 1475.98 -3354.2 1453.52
 -2336.4 1428.71  -399.6 1388.43   396.7 1395.52  1612.5 1390.35  2872.8 1369.11
  4028.2 1325.42 4386.36 1310.89  4936.2 1288.18    5424 1311.15    5429 1310.76
  5958.2 1349.26  6407.3 1354.42  7812.6 1363.79 11588.2 1372.23 13099.7 1406.37
   14253 1382.31 14613.6 1424.53 14896.9 1429.18 16731.6 1471.35   18052 1467.34
 19538.5 1466.74 20324.6 1474.22 21029.1 1532.61 21226.4 1532.13 21531.2 1528.55
#Mann= 20 ,-1 , 0
-10970.2      .1       0-10562.2      .1       0   -4927      .1       0
 -3354.2      .1       0 -2336.4     .16       0  -399.6     .16       0
   396.7      .1       0  1612.5      .1       0  4028.2      .1       0
 4386.36     .07       0    5429     .05       0  6407.3      .1       0
  7812.6      .1       0 13099.7      .1       0 14896.9      .1       0
 16731.6      .1       0   18052      .1       0 19538.5     .16       0
 20324.6      .1       0 21226.4      .1       0
Bank Sta=4386.36,5424
XS Rating Curve= 0 ,0
Exp/Cntr=0.3,0.1

Type RM Length L Ch R = 1 ,317742  ,1512,1512,1512
BEGIN DESCRIPTION:
PEDERNALES RIVER 257.0
END DESCRIPTION:
XS GIS Cut Line= 5
      2856323.79     10078660.44      2865238.41     10069445.89
      2866843.28     10061704.72      2864632.48     10055062.83
      2860170.79       10049331.
#Sta/Elev= 30
-11037.9 1532.98 -9078.1 1466.01 -6850.3 1437.54   -6292 1471.38 -5605.5 1491.19
 -4301.4 1463.87 -2446.5    1425  -901.8 1396.25  -129.7 1386.02   657.3 1375.59
  2888.6 1360.22 4454.55 1304.07  4908.1 1280.84  5439.2 1300.68    5455 1302.72
  5846.1  1340.9  6312.1 1341.29  7953.6 1342.65  9688.9 1355.48 11418.4 1329.67
 11995.8  1350.6 12664.4 1364.79 15170.9 1426.42 16452.3 1436.11 17903.3 1462.66
 19577.2 1425.79 20629.6 1473.28 22551.1 1484.43 23921.1 1536.45 23952.7 1537.12
#Mann= 20 ,-1 , 0
-11037.9      .1       0 -9078.1     .16       0   -6292      .1       0
 -4301.4      .1       0 -2446.5      .1       0  -901.8     .16       0
  -129.7      .1       0   657.3      .1       0  2888.6     .16       0
 4454.55     .07       0  5439.2      .1       0  5439.2      .1       0
  6312.1     .16       0  7953.6      .1       0 11995.8     .05       0
 12664.4      .1       0 16452.3      .1       0 20629.6      .1       0
 22551.1     .05       0 23921.1     .16       0
Bank Sta=4454.55,5455
XS Rating Curve= 0 ,0
Exp/Cntr=0.3,0.1

Type RM Length L Ch R = 1 ,316230  ,2038,2038,2038
BEGIN DESCRIPTION:
PEDERNALES RIVER 256.0
END DESCRIPTION:
XS GIS Cut Line= 4
      2857381.58     10079792.27      2867004.41     10069275.54
      2868924.93     10054161.53      2866899.15     10047292.72
#Sta/Elev= 30
-12369.8 1543.12-11477.1 1525.11   -7732 1451.27 -6781.7 1432.53 -2478.5  1393.9
  -532.8 1362.15   578.4 1362.26  1888.5 1374.21 4136.36 1308.57    4941  1277.5
  5344.4 1308.03  5404.9 1317.93    6563 1350.46  7362.8 1371.28  9704.7 1385.95
 11230.6 1397.85   13462 1404.75 14091.8 1367.17 15487.1 1392.93 15921.4 1418.09
 16311.3 1375.52 16631.2 1432.39 17329.4 1433.46 18598.6 1391.14 19620.5 1369.38
 20341.9 1386.55 20869.7  1377.6 21658.1 1435.79 23268.5 1475.42 24281.9 1539.31
#Mann= 19 ,-1 , 0
-12369.8      .1       0-11477.1      .1       0   -7732      .1       0
 -6781.7      .1       0 -2478.5      .1       0  -532.8      .1       0
   578.4      .1       0 4136.36     .07       0  5404.9      .1       0
    6563      .1       0  7362.8     .05       0  9704.7      .1       0
 11230.6      .1       0 15487.1      .1       0 17329.4     .16       0
 18598.6      .1       0 20341.9      .1       0 21658.1      .1       0
 23268.5      .1       0
Bank Sta=4136.36,5344.4
XS Rating Curve= 0 ,0
Exp/Cntr=0.3,0.1

Type RM Length L Ch R = 1 ,314192  ,1722,1722,1722
BEGIN DESCRIPTION:
PEDERNALES RIVER 260.0
END DESCRIPTION:
XS GIS Cut Line= 3
      2859013.12     10080403.31      2868125.91     10072024.59
      2872204.26     10053637.41
#Sta/Elev= 30
-12636.5 1516.48-11747.7 1491.95-10448.2 1458.82-10028.6 1453.28 -9681.5 1458.55
 -9369.8 1455.28   -7463 1435.27 -6559.5 1428.24  1249.9 1378.01  3377.3 1327.54
  4164.2 1303.25  4810.1 1276.35  5018.5 1273.19  5179.2 1274.22  5233.9 1286.03
  5548.3 1304.75  5553.4 1306.31  6873.7 1347.48  8126.9 1368.75  8578.4 1374.19
  8971.1 1378.92  9476.8 1385.01   10399 1396.11 11335.1 1407.38 12761.6 1426.67
   13426 1436.82 14057.6 1446.47 17738.7 1502.39 17928.4 1511.99 18576.8 1521.61
#Mann= 19 ,-1 , 0
-12636.5      .1       0-11747.7      .1       0-10448.2      .1       0
 -9369.8     .05       0   -7463      .1       0 -6559.5      .1       0
  1249.9      .1       0  4164.2     .07       0  5553.4      .1       0
  6873.7     .05       0  8126.9     .05       0  8578.4     .16       0
  8971.1      .1       0  9476.8     .05       0   10399     .05       0
 11335.1      .1       0 12761.6      .1       0   13426     .16       0
 14057.6      .1       0
Bank Sta=4164.2,5548.3
XS Rating Curve= 0 ,0
Exp/Cntr=0.3,0.1

Type RM Length L Ch R = 1 ,312470  ,1905,1905,1905
BEGIN DESCRIPTION:
PEDERNALES RIVER 262.0
END DESCRIPTION:
XS GIS Cut Line= 3
      2861305.79     10080327.06      2869687.59     10072095.73
      2874288.34     10053609.37
#Sta/Elev= 30
-11319.5 1513.82-11000.9  1504.1 -9899.1 1475.24 -8447.7  1464.7 -7279.5 1456.22
 -5566.2 1443.78   -4067  1432.9 -3416.5 1428.18 -2702.3 1475.36 -1512.2 1423.49
   646.7 1358.57    1859 1372.23  4665.7  1281.4  4727.5 1264.13  5015.8 1262.56
  5582.3  1284.4  5587.5 1283.75    6666 1299.38  7782.3 1332.57 11136.5  1376.6
 12136.8 1374.91 12750.3 1395.86 13297.3 1409.61   13974 1404.08 14803.3 1417.67
 15304.3 1429.27 17239.1 1448.23 17855.3 1470.14   18880 1496.18 19478.5 1531.74
#Mann= 19 ,-1 , 0
-11319.5     .16       0-11000.9      .1       0 -9899.1      .1       0
 -8447.7     .05       0 -7279.5      .1       0 -5566.2      .1       0
   -4067      .1       0 -1512.2      .1       0  4665.7     .07       0
  5582.3      .1       0    6666      .1       0 11136.5      .1       0
 12750.3      .1       0 13297.3     .16       0   13974      .1       0
 14803.3     .16       0 15304.3      .1       0 17239.1      .1       0
 17855.3      .1       0
Bank Sta=4665.7,5587.5
XS Rating Curve= 0 ,0
Exp/Cntr=0.3,0.1

Type RM Length L Ch R = 1 ,310565  ,2231,2231,2231
BEGIN DESCRIPTION:
PEDERNALES RIVER 264.0
END DESCRIPTION:
XS GIS Cut Line= 3
      2862596.85     10081228.29      2871404.24     10072272.92
      2875887.93      10054827.8
#Sta/Elev= 30
-11216.9 1511.48-10082.1 1457.87   -8377 1417.74 -6975.9 1418.35 -6347.4 1418.62
 -5561.3 1386.04 -3384.4 1382.56 -2394.6 1414.76 -1774.9 1398.42  -597.2 1389.84
     273 1363.92  1508.1 1323.19  2223.8 1322.51  4592.3 1270.71  4729.2 1249.51
  5225.1 1251.63  5442.6 1276.13  5817.3 1286.02  8648.9 1366.13  9528.5 1401.84
 10397.9 1385.05 11188.6 1420.59 11758.8 1436.16 13217.5 1438.91 13660.6 1426.33
 13763.9 1407.88 14153.8 1426.25 17773.1 1524.58 18417.8 1514.02 19355.8 1555.86
#Mann= 20 ,-1 , 0
-11216.9      .1       0-10082.1      .1       0   -8377      .1       0
 -6975.9     .16       0 -5561.3      .1       0 -3384.4     .16       0
 -1774.9      .1       0  -597.2     .16       0     273      .1       0
  2223.8      .1       0  4592.3     .07       0  5442.6      .1       0
  5817.3      .1       0  8648.9      .1       0  9528.5      .1       0
 11188.6     .16       0 11758.8      .1       0 13217.5      .1       0
 14153.8      .1       0 18417.8      .1       0
Bank Sta=4592.3,5442.6
XS Rating Curve= 0 ,0
Exp/Cntr=0.3,0.1
