HEC-RAS study PEDERNALES RIVER.prj: PEDERNALES RIVER Base Level Engineering

--- PEDERNALES RIVER.g02 (geometry) --- (continued)

Type RM Length L Ch R = 1 ,308334  ,2452,2452,2452
BEGIN DESCRIPTION:
PEDERNALES RIVER 266.0
END DESCRIPTION:
XS GIS Cut Line= 3
      2863528.56     10081708.37      2873277.75     10072399.95
      2877280.29     10055989.79
#Sta/Elev= 30
-10541.6 1524.33 -9575.8 1483.34 -7458.1 1417.99 -7044.2 1391.71 -6245.6 1400.01
 -4861.7 1358.46 -3684.5 1333.19 -3465.3 1357.08   -3235 1409.82 -2295.2 1369.49
 -1871.7 1349.37 -1364.7 1331.78  -405.3 1347.43    99.7 1343.16  1334.8    1326
  1817.5 1319.29  2232.9 1313.52  3594.4 1293.39  4476.9 1278.83  4482.1  1278.9
  4889.3  1234.6  5208.7 1241.26  5404.2 1271.85  5409.5 1274.29  6793.2 1304.38
   11793 1392.47 15095.7 1449.29 15548.4 1454.47 18158.5  1496.9   19829 1589.85
#Mann= 20 ,-1 , 0
-10541.6      .1       0 -9575.8      .1       0 -7458.1     .16       0
 -6245.6      .1       0 -4861.7      .1       0   -3235     .16       0
 -2295.2      .1       0 -1871.7     .16       0  -405.3      .1       0
    99.7      .1       0  1334.8      .1       0  1817.5     .16       0
  2232.9      .1       0  3594.4     .16       0  4476.9     .05       0
  5404.2     .16       0  6793.2      .1       0   11793      .1       0
 15095.7     .05       0 15548.4      .1       0
Bank Sta=4482.1,5409.5
XS Rating Curve= 0 ,0
Exp/Cntr=0.3,0.1

Type RM Length L Ch R = 1 ,305882  ,2222,2222,2222
BEGIN DESCRIPTION:
PEDERNALES RIVER 268.0
END DESCRIPTION:
XS GIS Cut Line= 3
      2863782.62     10082232.29      2876996.85     10070674.46
      2878048.13      10057092.9
#Sta/Elev= 30
 -9672.7 1514.74 -8461.9 1469.98 -6692.9 1404.69 -6092.2 1407.66 -5226.5 1371.22
 -4614.9 1371.51 -2823.2 1310.38 -2426.7 1348.22 -1931.1 1398.64  -128.5 1313.12
  1085.7 1328.84  1744.7 1323.27  3656.6  1276.7  4298.2 1245.47  4681.6 1254.14
  4922.2 1229.41  5254.9 1241.66    5291 1252.19  5489.4 1286.59  6042.8 1325.83
  7882.9 1359.72 10373.9 1366.53 11317.3 1370.09 12489.5  1385.4 13564.6 1407.34
   15481 1438.79 17275.8 1479.17 17942.3 1534.96 19357.7 1509.65 21505.1 1560.76
#Mann= 19 ,-1 , 0
 -9672.7      .1       0 -8461.9      .1       0 -6092.2     .16       0
 -4614.9      .1       0 -2426.7      .1       0  -128.5      .1       0
  1085.7      .1       0  1744.7     .16       0  3656.6      .1       0
  4681.6     .05       0  5254.9      .1       0  6042.8      .1       0
 10373.9     .05       0 11317.3      .1       0 12489.5     .16       0
 13564.6     .16       0   15481      .1       0 17275.8      .1       0
 19357.7      .1       0
Bank Sta=4681.6,5291
XS Rating Curve= 0 ,0
Exp/Cntr=0.3,0.1

Type RM Length L Ch R = 1 ,303660  ,2431,2431,2431
BEGIN DESCRIPTION:
PEDERNALES RIVER 269.0
END DESCRIPTION:
XS GIS Cut Line= 3
      2864141.38     10082705.47      2872717.58     10075622.38
      2881513.83     10071823.58
#Sta/Elev= 30
 -8372.6 1516.19 -6991.7 1463.89 -3365.9 1351.59   -2782 1348.87 -2555.7 1344.32
 -1127.7 1296.71  -926.8 1309.15  -283.2 1364.19   473.3 1331.06  1320.6  1296.9
  1636.8  1292.8  2167.5    1289  2803.8 1302.37  3807.9  1257.1  4159.5 1252.18
    4418 1247.62  4429.3  1246.7  4826.9 1224.99  5245.8 1242.34  5253.9 1246.66
  5382.4 1275.31  5528.4 1273.81  6241.4 1263.22  6868.9 1331.28  7672.2  1356.7
  9344.8 1354.32  9764.7 1377.07 10578.2 1420.19 11138.8 1405.58 12331.9 1446.43
#Mann= 19 ,-1 , 0
 -8372.6      .1       0 -6991.7      .1       0   -2782     .16       0
 -2555.7      .1       0  -926.8     .16       0  -283.2      .1       0
   473.3     .16       0  1320.6      .1       0  1636.8     .16       0
  2167.5      .1       0  2803.8     .16       0  3807.9      .1       0
  4159.5     .16       0  4429.3     .05       0  5245.8      .1       0
  5528.4      .1       0  6868.9      .1       0  7672.2      .1       0
  9764.7      .1       0
Bank Sta=4418,5253.9
XS Rating Curve= 0 ,0
Exp/Cntr=0.3,0.1

Type RM Length L Ch R = 1 ,301229  ,1762,1762,1762
BEGIN DESCRIPTION:
Mapping XS 468fd7d0
END DESCRIPTION:
XS GIS Cut Line= 4
      2864500.23     10083178.58      2872128.84     10076917.32
      2876034.62     10076964.99      2881392.54     10073228.48
#Sta/Elev= 30
   -6606 1485.26 -6018.7    1465 -5634.9 1461.03 -4941.3 1451.38   -3694 1418.64
  -924.2 1339.98  -594.5 1332.23  -237.6 1330.49   353.4 1306.92   940.9 1294.71
  1127.3  1289.1  1357.8 1315.68  1943.2 1325.04  2927.4 1300.26  3362.7 1275.93
  3562.7 1268.63  3942.6 1274.38    4203 1256.17  4542.8    1226  5012.5 1215.52
 5596.59  1256.7  5884.7 1278.36  6617.6 1303.85  7168.6 1323.02  7856.2 1301.43
  8256.7 1319.15  9192.5 1352.11 10606.2 1373.16 11964.6 1443.13 13701.3 1452.28
#Mann= 19 ,-1 , 0
   -6606      .1       0 -6018.7     .05       0 -5634.9      .1       0
 -4941.3      .1       0   -3694      .1       0  -924.2      .1       0
  -594.5     .16       0   353.4      .1       0   940.9     .16       0
  1357.8      .1       0  2927.4      .1       0  3362.7      .1       0
  3942.6      .1       0    4203     .05       0 5596.59     .16       0
  5884.7     .16       0  6617.6      .1       0  8256.7      .1       0
  9192.5      .1       0
Bank Sta=4203,5596.59
XS Rating Curve= 0 ,0
Exp/Cntr=0.3,0.1

Type RM Length L Ch R = 1 ,299467  ,1509,1509,1509
BEGIN DESCRIPTION:
Mapping XS b7bac6b9
END DESCRIPTION:
XS GIS Cut Line= 4
      2864912.37     10083548.22      2871432.78     10078471.37
      2875859.31     10078525.39      2881013.38     10074318.72
#Sta/Elev= 30
 -4933.2    1452 -4873.8 1450.14   -3304 1446.44 -2688.2 1446.84  -557.4 1366.24
   922.4 1326.37  1237.7 1327.33    1273 1310.31  1360.9 1307.16  1564.7  1301.2
  2179.7  1280.1    2731 1286.21  3229.7 1267.52  3318.7 1280.61  3605.1 1270.77
  4149.4 1251.83  4616.4 1253.47  4686.4 1234.49  4746.4 1216.75  5046.2 1213.05
 5477.27 1236.05  5678.7 1249.68  6332.7 1290.39  7004.6 1314.55  7572.7 1334.34
  7953.6 1346.79  9201.4 1356.21    9912 1339.52 12257.1 1410.85 14410.3 1455.82
#Mann= 18 ,-1 , 0
 -4933.2     .05       0 -4873.8     .05       0   -3304      .1       0
   922.4     .05       0  1360.9     .16       0  1564.7      .1       0
  2179.7      .1       0    2731      .1       0  3229.7     .16       0
  3605.1      .1       0  4149.4     .16       0  4686.4     .05       0
 5477.27      .1       0  5678.7      .1       0  6332.7     .16       0
  7004.6      .1       0  7572.7      .1       0  7953.6      .1       0
Bank Sta=4686.4,5477.27
XS Rating Curve= 0 ,0
Exp/Cntr=0.3,0.1

Type RM Length L Ch R = 1 ,297958  ,1286,1286,1286
BEGIN DESCRIPTION:
Mapping XS 5d83a6b7
END DESCRIPTION:
XS GIS Cut Line= 4
      2865533.48     10083868.29      2871206.05     10079979.05
      2875841.51     10079983.54      2880952.96     10075098.31
#Sta/Elev= 30
 -3603.8 1426.52 -3481.7 1420.12   -3005 1430.83 -2252.1 1415.63 -1432.9 1431.35
 -1201.3 1435.63  -108.8 1393.48   619.6    1368  1428.6 1353.61    1611 1334.28
  2015.6 1315.93  2414.8 1296.86    4150 1233.69  4546.4 1216.02  4666.4 1232.21
  4756.4 1216.47  4906.2 1210.05 5590.91 1232.23  5915.3 1247.01  6860.8 1290.07
  7268.2 1308.85  7889.7 1337.51  8791.1 1335.11  8982.4 1349.34  9182.5 1349.33
  9540.9  1352.2 10432.3 1382.65 12905.5 1413.32 13574.1 1421.68   14980 1440.37
#Mann= 19 ,-1 , 0
 -3603.8     .16       0   -3005      .1       0 -2252.1     .16       0
 -1432.9      .1       0  -108.8      .1       0   619.6      .1       0
  1428.6     .16       0  2015.6      .1       0  2414.8      .1       0
    4150      .1       0  4666.4     .05       0 5590.91      .1       0
  5915.3      .1       0  6860.8     .16       0  7268.2      .1       0
  7889.7      .1       0  9182.5      .1       0 12905.5      .1       0
 13574.1      .1       0
Bank Sta=4666.4,5590.91
XS Rating Curve= 0 ,0
Exp/Cntr=0.3,0.1

Type RM Length L Ch R = 1 ,296672  ,1216,1216,1216
BEGIN DESCRIPTION:
Mapping XS 632ee251
END DESCRIPTION:
XS GIS Cut Line= 4
      2866049.23     10084291.22      2871601.69     10081702.67
      2878501.88     10079651.43      2880891.13     10075930.51
#Sta/Elev= 30
 -2953.4 1435.02 -2198.7  1404.5 -2068.8 1396.59 -1548.5 1414.21   -1255 1421.68
  -538.5  1439.9  1613.6 1321.43  1711.1 1304.23  1790.7  1312.4  3172.8 1287.12
  4442.2    1243  4713.5 1224.97  4796.3 1208.64  4932.3 1205.65  5495.2 1225.04
  6126.5 1252.93  6537.9 1281.38  6820.9 1305.05  7227.7 1338.03    7412 1343.06
  8267.5 1341.61  9428.4 1332.13  9597.4 1332.76 10374.5 1361.24 10816.5  1364.7
 11877.4 1337.21 12198.8 1336.18 12752.8 1353.68 13906.8 1387.34 14793.4 1433.44
#Mann= 16 ,-1 , 0
 -2953.4     .16       0 -2198.7     .05       0 -2068.8      .1       0
 -1548.5     .16       0   -1255      .1       0  4713.5     .05       0
  5495.2      .1       0  6126.5      .1       0  6537.9     .16       0
  6820.9     .16       0    7412      .1       0  8267.5      .1       0
  9428.4     .16       0  9597.4      .1       0 11877.4     .16       0
 12752.8      .1       0
Bank Sta=4713.5,5495.2
XS Rating Curve= 0 ,0
Exp/Cntr=0.3,0.1

Type RM Length L Ch R = 1 ,295456  ,1418,1418,1418
BEGIN DESCRIPTION:
Mapping XS 9e6836ef
END DESCRIPTION:
XS GIS Cut Line= 3
      2867714.99     10084363.64      2880162.61     10080140.47
      2881359.12     10075988.56
#Sta/Elev= 30
 -1550.2 1434.33  -120.9  1412.1  2104.3 1293.15  2554.1    1272  3701.7 1243.87
  3972.6 1254.44  4324.8 1222.02  4683.8 1222.42  4689.5 1220.47  4799.9 1198.83
  5034.7 1197.51  5180.1  1203.2  5280.9 1225.15  5733.5  1247.8  6486.1 1276.13
  6755.1 1290.75  7596.7 1289.16  7763.9 1295.95  8237.7 1295.75  8520.3 1314.12
  8790.4 1318.53  9731.3 1337.57 10240.3 1333.69 10557.5 1331.31 11596.8 1293.81
 12286.8 1289.35 12538.1 1304.02 13636.5 1367.85 14316.6 1373.95 15915.2 1422.15
#Mann= 19 ,-1 , 0
 -1550.2      .1       0  2104.3     .16       0  2554.1      .1       0
  4689.5     .05       0  5280.9     .16       0  5733.5      .1       0
  6486.1      .1       0  6755.1     .16       0  7596.7     .16       0
  7763.9      .1       0  8520.3     .16       0  8790.4      .1       0
  9731.3      .1       0 10240.3     .16       0 10557.5      .1       0
 12286.8     .16       0 12538.1      .1       0 13636.5      .1       0
 14316.6      .1       0
Bank Sta=4683.8,5280.9
XS Rating Curve= 0 ,0
Exp/Cntr=0.3,0.1

Type RM Length L Ch R = 1 ,294038  ,1420,1420,1420
BEGIN DESCRIPTION:
Mapping XS 98904cda
END DESCRIPTION:
XS GIS Cut Line= 4
       2868067.1     10084671.76      2873282.73     10084084.33
      2880570.32     10080874.63      2881942.21     10075162.07
#Sta/Elev= 30
 -1598.3 1409.27    -682 1389.68   122.6 1403.81   818.2 1358.09  2271.6 1318.76
  3845.4 1229.99    3965 1243.38  4214.7 1231.68  4482.2 1248.43  4685.3 1227.64
  4755.3  1202.6  5051.4 1196.08  5400.1 1224.08  5423.5 1224.55  5678.6 1249.43
  6582.6 1250.79  7015.8 1232.94    7742 1234.57  8342.7 1302.09  8900.4 1308.66
  9607.4 1268.83  9914.2 1266.96 10140.6 1295.99 10738.1  1285.9   11059 1269.92
 11440.3 1259.56 11692.3 1264.35 13233.8  1301.8 14258.7 1361.82 17488.4 1422.12
#Mann= 17 ,-1 , 0
 -1598.3      .1       0  3845.4     .16       0    3965     .16       0
  4685.3     .05       0  5400.1      .1       0  6582.6     .16       0
  7015.8      .1       0    7742     .16       0  8342.7      .1       0
  8900.4     .16       0  9607.4      .1       0 10738.1     .16       0
   11059     .16       0 11440.3     .16       0 11692.3      .1       0
 13233.8      .1       0 14258.7      .1       0
#XS Ineff= 2 , 0
                         6463.07         1256.63
Permanent Ineff=
       F       F
Bank Sta=4685.3,5423.5
XS Rating Curve= 0 ,0
Exp/Cntr=0.3,0.1

Type RM Length L Ch R = 1 ,292618  ,1397,1397,1397
BEGIN DESCRIPTION:
Mapping XS cafbb9bf
END DESCRIPTION:
XS GIS Cut Line= 5
       2869842.2     10085040.64      2873520.87     10085910.18
      2878379.79     10082540.62      2881132.89     10081011.71
      2882824.48     10074000.95
#Sta/Elev= 30
 -1206.6 1418.82   258.5    1364  1050.5 1365.68  1708.6 1311.99  2108.6 1288.89
  2326.9 1307.26  2820.1 1317.87  3191.4 1296.45  3489.9 1280.24  4081.9 1246.26
  4810.2  1213.4  4818.9 1212.03  5054.5 1187.58  5415.4 1211.06  5436.4  1212.4
  5634.6 1226.59  6161.2 1262.48  6833.9 1237.91  7413.5 1209.62  7835.7 1256.15
  8174.2 1280.01  9148.9 1254.56 10951.3 1241.18 11851.4 1258.97 12786.5 1278.83
 13501.8 1306.41 14279.1 1344.85 14896.3 1351.37 15254.9 1358.82 18847.5 1427.68
#Mann= 20 ,-1 , 0
 -1206.6      .1       0  1708.6      .1       0  2326.9      .1       0
  2820.1      .1       0  3191.4      .1       0  3489.9     .16       0
  4081.9      .1       0  4818.9     .05       0  5415.4      .1       0
  5634.6      .1       0  6833.9     .16       0  7835.7      .1       0
  9148.9      .1       0 10951.3      .1       0 11851.4      .1       0
 12786.5      .1       0 13501.8      .1       0 14279.1      .1       0
 14896.3     .16       0 15254.9      .1       0
#XS Ineff= 2 , 0
                         6193.18         1263.39
Permanent Ineff=
       F       F
Bank Sta=4810.2,5436.4
XS Rating Curve= 0 ,0
Exp/Cntr=0.3,0.1

Type RM Length L Ch R = 1 ,291221  ,1740,1740,1740
BEGIN DESCRIPTION:
Mapping XS 4bb0072c
END DESCRIPTION:
XS GIS Cut Line= 5
      2871492.99     10085989.61      2875304.21     10086665.47
      2878272.98     10083468.15      2881708.81     10081122.92
      2882816.62     10075710.92
#Sta/Elev= 30
 -1066.8 1396.68      17 1335.44   470.9 1311.05   980.1 1340.84  1368.5 1302.02
    1734 1285.92  2252.3  1337.8  2969.9 1309.04  3637.3 1268.95  4683.3 1246.66
  4817.6 1224.31    4825 1194.82  4839.1 1183.47  5022.6 1181.61  5716.2 1223.67
  6295.5 1245.58  6928.7 1209.86  7493.6 1210.62  7857.7 1207.74  8380.4 1239.54
  9368.1 1230.35  9909.6 1220.25 10791.3 1270.88   11704 1304.24 12193.2 1279.69
 12876.3 1286.14 13300.5 1299.48 13919.3 1326.36 14818.9 1344.65 16851.1 1386.59
#Mann= 19 ,-1 , 0
 -1066.8      .1       0      17      .1       0  1368.5      .1       0
    1734     .16       0  2969.9      .1       0  3637.3      .1       0
  4817.6     .05       0  5716.2     .16       0  6295.5      .1       0
  6295.5     .16       0  6928.7      .1       0  7493.6      .1       0
  8380.4      .1       0  9368.1      .1       0 10791.3      .1       0
 12876.3     .16       0 13300.5      .1       0 13919.3      .1       0
 14818.9      .1       0
#XS Ineff= 2 , 0
                            6250         1249.19
Permanent Ineff=
       F       F
Bank Sta=4817.6,5716.2
XS Rating Curve= 0 ,0
Exp/Cntr=0.3,0.1

Type RM Length L Ch R = 1 ,289481  ,1914,1914,1914
BEGIN DESCRIPTION:
Mapping XS 0e9bef21
END DESCRIPTION:
XS GIS Cut Line= 5
      2877801.37     10088323.55      2878682.34     10083711.87
      2879430.69     10082852.94      2882077.68     10081127.42
      2882866.06     10076992.02
#Sta/Elev= 30
  1427.8 1316.48  2076.3 1289.37  2622.6 1306.53  4422.6 1251.94  4575.4 1241.92
  4756.7 1209.59  4777.1 1193.59  4960.7  1179.3  5330.7 1187.66  5591.2 1210.81
  5596.3 1210.23  5795.2 1218.41  6225.5 1187.93  6520.1 1197.99  6794.6    1199
  6955.3 1206.27  7194.9 1241.61  8640.7 1213.09  9161.6 1261.48  9262.3 1277.58
  9631.2 1287.77   10457 1333.59 11197.2 1295.63 11852.2 1300.56 12052.4 1303.65
 12143.4  1306.9 12529.7 1319.78 12787.4  1317.2 14030.5 1356.95 14631.7 1370.68
#Mann= 18 ,-1 , 0
  1427.8      .1       0  2622.6      .1       0  4422.6     .16       0
  4575.4      .1       0  4777.1     .05       0  5591.2     .16       0
  6520.1      .1       0  6794.6      .1       0  6955.3     .16       0
  7194.9      .1       0  9161.6     .16       0  9631.2      .1       0
 11852.2     .16       0 12052.4     .16       0 12143.4      .1       0
 12529.7      .1       0 12787.4     .16       0 14030.5      .1       0
#XS Ineff= 2 , 0
                         7272.73         1243.55
Permanent Ineff=
       F       F
Bank Sta=4756.7,5596.3
XS Rating Curve= 0 ,0
Exp/Cntr=0.3,0.1

Type RM Length L Ch R = 1 ,287567  ,847,847,847
BEGIN DESCRIPTION:
Mapping XS 5d15e5cf
END DESCRIPTION:
XS GIS Cut Line= 4
       2878539.1     10088332.59      2879424.83     10085109.85
      2879418.64     10082950.45      2882841.18     10080809.03
#Sta/Elev= 30
  -185.5 1304.71   324.1 1291.56   773.5 1303.83  1455.3  1287.2    2280  1256.3
  3149.6 1236.84  3484.7 1215.86  3672.9 1201.44  3862.9 1182.59  4072.9 1184.26
  4962.6 1170.66  5052.9 1173.29  5072.9 1182.02  5092.9 1198.16  5112.9 1217.88
  5122.9 1223.01  5324.8 1241.39  6619.8  1211.1  6743.3 1213.42  7120.7 1236.23
  7216.7  1254.7  7228.8 1256.33  7295.4 1273.25  7462.6 1286.68  7629.6 1292.83
    7998 1300.81  8652.4 1350.65    8945    1351  8973.9 1350.66  9353.4 1342.09
#Mann= 11 ,-1 , 0
  -185.5      .1       0  3484.7     .16       0  3672.9     .05       0
  5092.9     .16       0  5324.8      .1       0  7216.7     .16       0
  7228.8      .1       0  7462.6     .16       0  7629.6      .1       0
    8945     .16       0  8973.9      .1       0
#XS Ineff= 2 , 0
                         5343.18         1241.99
Permanent Ineff=
       F       F
Bank Sta=3672.9,5092.9
XS Rating Curve= 0 ,0
Exp/Cntr=0.3,0.1

Type RM Length L Ch R = 1 ,286720  ,985,985,985
BEGIN DESCRIPTION:
Mapping XS 2efcf93c
END DESCRIPTION:
XS GIS Cut Line= 3
      2880217.95     10088166.49      2880248.95     10082784.81
      2882644.43     10081321.56
#Sta/Elev= 30
   185.8 1284.13   874.4 1251.42  1158.3 1237.13  1578.5 1227.74  1593.4 1227.74
  2348.6 1241.92  2908.6 1231.29  3264.6 1244.72  3596.9 1246.88  3848.6 1239.49
  4358.6 1192.09  4478.6 1178.06  4848.6 1182.98  5028.4 1169.24  5078.6 1173.49
  5108.6 1195.89  5138.6 1208.46  5248.6 1222.31  5548.6 1223.74  6077.4 1199.37
  6335.2  1213.1  6404.5 1219.77  6578.7 1233.15  6630.9 1246.13  6656.5 1262.36
    6689 1277.22  6775.3 1291.12  7575.5 1324.02  8034.2 1364.56  8374.6 1365.55
#Mann= 14 ,-1 , 0
   185.8      .1       0   874.4     .16       0  1158.3      .1       0
  1578.5     .05       0  1593.4      .1       0  3264.6     .16       0
  3596.9      .1       0  4358.6     .05       0  5108.6     .16       0
  5548.6      .1       0  6335.2     .16       0  6404.5      .1       0
  6656.5     .16       0  6775.3      .1       0
#XS Ineff= 2 , 0
                         5426.14         1226.66
Permanent Ineff=
       F       F
Bank Sta=4358.6,5108.6
XS Rating Curve= 0 ,0
Exp/Cntr=0.3,0.1

Type RM Length L Ch R = 1 ,285735  ,863,863,863
BEGIN DESCRIPTION:
Mapping XS bbd2c49a
END DESCRIPTION:
XS GIS Cut Line= 3
      2881152.35     10088420.92      2881226.14     10082380.07
      2882675.01     10081617.28
#Sta/Elev= 30
  -232.5    1281   474.7 1254.39   883.7 1269.09  1296.9 1267.27  1478.4 1262.73
  1617.6 1262.36  2004.9 1264.65  2354.9 1251.63  3054.9 1194.61  3204.9 1204.55
    3385 1230.97    3675 1245.79    4255 1222.66  4635.1 1189.21  4770.7 1171.84
  5034.8 1168.29  5155.1 1177.33  5225.1 1170.85  5395.1 1188.31  5475.1 1205.78
  5775.1 1233.13  5852.8 1254.69  5890.5 1282.73  5969.7 1295.71  6408.7 1322.65
    6450 1324.36  6712.7 1334.38  6732.2 1335.06  7235.4 1374.47  7446.2 1375.21
#Mann= 13 ,-1 , 0
  -232.5      .1       0   883.7     .16       0  1296.9      .1       0
  1478.4     .16       0  1617.6      .1       0  2354.9      .1       0
  4635.1     .05       0  5395.1      .1       0  5852.8     .16       0
  6408.7     .16       0    6450      .1       0  6712.7     .16       0
  6732.2      .1       0
#XS Ineff= 2 , 0
         3681.82 1246.37
Permanent Ineff=
       F       F
Bank Sta=4635.1,5395.1
XS Rating Curve= 0 ,0
Exp/Cntr=0.3,0.1

Type RM Length L Ch R = 1 ,284872  ,1035,1035,1035
BEGIN DESCRIPTION:
Mapping XS 5be24633
END DESCRIPTION:
XS GIS Cut Line= 3
      2881935.19     10088291.62      2882057.88     10082511.76
      2882708.21     10081859.97
#Sta/Elev= 30
    87.1 1300.68   749.5 1295.01  1002.7 1294.44  1146.3 1293.69  1297.5 1294.74
  1395.8 1296.66  1721.1 1286.83  2075.4 1256.82  2459.4 1252.72  2561.8 1250.66
  3303.4 1223.04  3406.4 1215.28  3754.4 1181.86  3848.5 1194.06  4215.9 1207.02
    4666 1187.85    4676 1187.31    4786 1166.83  4955.8 1164.14  5190.2 1170.09
  5246.2 1182.19  5286.2 1203.41  5376.2 1229.61  5576.2 1251.35  5646.2 1265.13
  5706.3 1308.64  5771.1 1317.15    6033 1344.23  6264.3 1357.08    6789 1382.16
#Mann= 18 ,-1 , 0
    87.1      .1       0   749.5      .1       0  1002.7     .16       0
  1146.3      .1       0  1297.5     .16       0  1395.8      .1       0
  1721.1      .1       0  2459.4     .05       0  2561.8      .1       0
  3303.4     .16       0  3406.4      .1       0  3754.4     .16       0
  3848.5      .1       0    4666     .05       0  5246.2      .1       0
  5771.1      .1       0    6033     .16       0  6264.3      .1       0
Bank Sta=4676,5246.2
XS Rating Curve= 0 ,0
Exp/Cntr=0.3,0.1

Type RM Length L Ch R = 1 ,283837  ,1169,1169,1169
BEGIN DESCRIPTION:
Mapping XS a3bec1fe
END DESCRIPTION:
XS GIS Cut Line= 3
      2882474.16     10088228.69      2882588.76     10084532.17
      2883294.45     10082146.86
#Sta/Elev= 30
   919.3 1292.74  1260.1 1269.68  1436.7 1257.52  1914.7 1237.84  2160.5 1237.62
  2259.3 1243.83  2655.1 1263.76  3035.3 1262.11  3415.5 1246.43  4015.7    1200
  4355.9 1183.06  4415.9 1189.64    4486 1186.61    4606 1169.19  4632.9 1173.05
  5147.6 1164.21  5201.7 1178.13 5213.64 1185.36  5241.7 1220.54  5273.4 1230.57
  5309.4  1232.4    5408 1246.33  5721.4 1276.87  5793.3 1298.44  5804.8 1311.13
    5837 1325.85    5942 1338.48  6538.8 1362.87  6958.9 1394.22  7105.1  1394.9
#Mann= 9 ,-1 , 0
   919.3      .1       0  1260.1     .16       0  1436.7      .1       0
  2160.5     .16       0  2259.3      .1       0    4486     .05       0
  5201.7     .05       0  5309.4     .16       0    5408      .1       0
Bank Sta=4486,5213.64
XS Rating Curve= 0 ,0
Exp/Cntr=0.3,0.1

Type RM Length L Ch R = 1 ,282668  ,1542,1542,1542
BEGIN DESCRIPTION:
Mapping XS a81cf08a
END DESCRIPTION:
XS GIS Cut Line= 4
      2883165.11     10088514.96      2882969.99     10086012.54
      2883976.65     10083194.93      2883934.97      10082343.7
#Sta/Elev= 30
  1609.8 1317.83  2400.6 1282.74  2894.9 1286.57  3035.3  1282.4  3406.5 1253.75
  3650.6 1222.39  3807.7 1209.51    3937  1213.6  4306.4  1227.8  4424.3 1214.55
  4522.1 1197.34  4690.8 1179.55  4783.1 1162.03  4829.8 1160.27  5254.5 1165.15
  5285.3 1171.27  5321.4 1193.28  5329.1 1196.74  5425.3 1205.67  5517.8 1211.69
  5733.9 1220.04  5836.8 1228.16  6160.9 1247.73  6628.4 1259.68  6826.4 1271.21
  6920.4 1284.23  7071.1 1295.04  7743.8  1369.9  7912.3 1381.77  7964.1 1383.62
#Mann= 13 ,-1 , 0
  1609.8      .1       0  3650.6     .16       0    3937      .1       0
  4424.3     .16       0  4522.1     .05       0  5321.4      .1       0
  5425.3     .16       0  5517.8      .1       0  5733.9     .16       0
  5836.8      .1       0  6160.9     .16       0  7071.1      .1       0
  7912.3     .16       0
Bank Sta=4522.1,5329.1
XS Rating Curve= 0 ,0
Exp/Cntr=0.3,0.1

Type RM Length L Ch R = 1 ,281126  ,1041,1041,1041
BEGIN DESCRIPTION:
Mapping XS 92669579
END DESCRIPTION:
XS GIS Cut Line= 3
      2883780.87     10088703.06      2884426.92     10086981.74
      2884441.25     10082398.63
#Sta/Elev= 30
  2268.7 1315.32    2506 1298.76  2676.9 1297.43  3018.5 1303.54  3239.2 1296.44
    3531 1280.89  4245.3 1264.55  4405.3 1252.73  4745.3  1207.9  4785.3 1197.75
  4805.3 1186.27  4835.3 1157.45    4875 1151.87  5135.3 1153.35  5285.3 1175.98
  5390.5 1185.38  5565.3 1202.25  5769.9 1214.93  6205.9 1236.73  6756.7 1251.53
  6847.8 1253.71  6866.4 1254.34  7315.3 1271.15  7375.3 1278.35  7635.3 1294.16
  7905.3 1321.54  8155.3 1338.01  8295.3 1351.51  8575.3 1369.53  8690.4 1370.88
#Mann= 8 ,-1 , 0
  2268.7      .1       0  4805.3     .05       0  5390.5      .1       0
  5390.5     .16       0  5769.9      .1       0  6756.7     .16       0
  6847.8      .1       0  6866.4     .16       0
Bank Sta=4805.3,5390.5
XS Rating Curve= 0 ,0
Exp/Cntr=0.3,0.1

Type RM Length L Ch R = 1 ,278510  ,1159,1159,1159
BEGIN DESCRIPTION:
Mapping XS 6115e061
END DESCRIPTION:
XS GIS Cut Line= 3
      2885936.27     10089625.26      2887039.59     10087992.85
      2886938.13     10082658.51
#Sta/Elev= 30
  1503.1 1317.33  1786.2 1313.72  2031.9 1323.66  2243.6  1320.6  2442.5 1315.89
  2557.9 1313.05  2926.8 1294.83  3130.1  1280.1  3399.7 1263.27  3670.5 1257.87
  4324.5 1214.16  4412.7 1212.65  4732.7 1188.18  4802.8 1173.25  4832.8 1156.33
  4872.8    1150  5102.6 1147.37  5375.5 1176.07  5659.3 1188.76  5833.7 1200.02
  6011.7 1211.55  6213.5 1223.18  6563.1 1236.96  6743.1 1252.46  6873.2 1270.19
  7103.2 1289.58  7279.6 1297.11  7933.3 1336.55  8373.4 1334.74  8808.7 1341.56
#Mann= 17 ,-1 , 0
  1503.1      .1       0  2243.6     .16       0  2442.5      .1       0
  2557.9      .1       0  2926.8     .16       0  3130.1     .16       0
  3399.7      .1       0  3670.5      .1       0  4324.5      .1       0
  4802.8     .05       0  5375.5     .16       0  5659.3      .1       0
  5833.7     .16       0  6011.7      .1       0  6213.5      .1       0
  6873.2     .16       0  7279.6      .1       0
Bank Sta=4802.8,5375.5
XS Rating Curve= 0 ,0
Exp/Cntr=0.3,0.1

Type RM Length L Ch R = 1 ,277351  ,1593,1593,1593
BEGIN DESCRIPTION:
Mapping XS 9b352956
END DESCRIPTION:
XS GIS Cut Line= 3
      2887001.43      10089409.1      2888198.51     10086923.67
      2887915.76     10082796.93
#Sta/Elev= 30
  1804.6 1264.18  2067.1 1257.07  2451.7 1269.64  2641.5 1257.61  2939.1 1241.72
  3019.4 1233.48  3031.5  1231.9    3243 1206.07  3395.8 1221.79    3546 1221.89
  3567.4 1223.79  3674.4 1225.61  3708.7 1223.69  3842.3 1212.45  4102.2 1219.54
  4418.9 1206.52  4637.7 1190.39  4773.7 1172.53  4833.9 1147.26    4994 1145.79
  5094.5 1146.95  5364.3 1173.83  5375.1 1174.66  5817.7    1205  6340.4 1234.21
  6427.6  1272.8  6542.8 1288.85  6684.2 1301.29  7159.3  1321.4  8699.7 1341.69
#Mann= 15 ,-1 , 0
  1804.6      .1       0  2641.5     .16       0  2939.1      .1       0
  3019.4     .16       0  3031.5      .1       0    3546     .16       0
  3567.4      .1       0  3674.4     .16       0  3708.7      .1       0
  4102.2     .16       0  4773.7     .05       0  5375.1     .16       0
  5817.7      .1       0  6340.4     .16       0  6542.8      .1       0
Bank Sta=4773.7,5364.3
XS Rating Curve= 0 ,0
Exp/Cntr=0.3,0.1

Type RM Length L Ch R = 1 ,271627  ,1630,1630,1630
BEGIN DESCRIPTION:
Mapping XS 20aac99c
END DESCRIPTION:
XS GIS Cut Line= 2
      2895204.11     10088176.03      2891361.63     10082108.13
#Sta/Elev= 30
    1950 1334.71    2014 1332.38  2930.1 1284.16  3097.3 1279.01  3290.3 1273.56
  3609.3 1258.33  3933.7 1232.25  3976.7 1216.93  4137.1 1197.53  4205.4 1189.75
  4580.4 1160.73  4586.5 1158.74  4789.9  1137.2  4983.7  1133.2  5093.3 1134.18
  5123.9 1143.97  5223.9 1148.37  5266.9 1162.69  5333.2 1180.21  5635.5 1208.06
  5834.1 1220.28    6435 1219.66  6566.5  1238.5  6783.1 1255.76    6859 1258.39
  8216.9 1283.21  8536.9 1288.69  8702.9 1290.38    8809 1291.46  9132.2 1294.75
#Mann= 18 ,-1 , 0
    1950     .16       0    2014      .1       0  2930.1     .16       0
  3097.3      .1       0  3290.3     .16       0  3933.7      .1       0
  4137.1     .16       0  4205.4      .1       0  4586.5     .05       0
  5266.9      .1       0  5635.5     .16       0  6566.5      .1       0
  6783.1     .16       0    6859      .1       0  8216.9     .16       0
  8536.9      .1       0  8702.9     .16       0    8809      .1       0
Bank Sta=4580.4,5266.9
XS Rating Curve= 0 ,0
Exp/Cntr=0.3,0.1

Type RM Length L Ch R = 1 ,269997  ,1738,1738,1738
BEGIN DESCRIPTION:
Mapping XS 833a2dfa
END DESCRIPTION:
XS GIS Cut Line= 3
      2896874.13     10087904.81      2893666.93      10082698.8
       2891699.9     10081758.38
#Sta/Elev= 30
  1554.1 1317.71    1658 1315.27  2004.4 1303.07  2254.4 1288.85  2847.5 1283.31
  3026.4  1284.2  3203.4  1275.8  3672.4 1258.88  3762.3 1256.26  4174.6 1229.76
  4325.8 1210.64  4546.6  1167.6  4647.1 1143.27  4967.5 1133.05  5083.6 1136.07
  5114.2  1144.8  5199.6 1143.87  5330.9 1166.22  5556.9 1191.67    5813 1199.68
  5941.3 1207.42  6515.1 1213.66  6880.5 1232.75  7243.2 1239.56  8175.1 1257.66
  8900.3 1259.48  9038.5 1265.01  9144.3 1268.01  9251.5 1270.06    9849 1279.82
#Mann= 17 ,-1 , 0
  1554.1      .1       0    1658     .16       0  2004.4     .16       0
  2254.4      .1       0  2847.5     .16       0  3203.4      .1       0
  3672.4     .16       0  3762.3      .1       0  4325.8      .1       0
  4546.6     .05       0  5330.9     .16       0    5813      .1       0
  6880.5     .16       0  7243.2      .1       0  9038.5     .16       0
  9144.3      .1       0  9251.5     .16       0
Bank Sta=4546.6,5330.9
XS Rating Curve= 0 ,0
Exp/Cntr=0.3,0.1

Type RM Length L Ch R = 1 ,268259  ,1359,1359,1359
BEGIN DESCRIPTION:
Mapping XS 9c8e1187
END DESCRIPTION:
XS GIS Cut Line= 5
      2898985.12     10087347.26      2897123.72     10084532.79
      2894669.09     10082523.56      2893193.68     10082213.84
      2891349.42     10081399.59
#Sta/Elev= 30
     834 1309.06  1115.5 1295.75  1287.1 1289.24  1955.7 1267.91    2270 1255.63
  2935.2 1255.53  3092.2 1253.35    3688 1242.91  3803.8 1240.12  4148.4 1228.94
  4588.5  1193.1  4751.5 1164.57  4757.9 1158.78  4780.2 1132.82  4794.5 1127.26
  4964.4 1125.98  5326.5 1139.37  5455.6 1153.71  5705.9 1166.48  6584.2  1200.2
  6833.7 1216.71  7060.7 1219.29    7216 1217.85  8182.9 1210.97  8899.9 1246.79
  9423.2 1237.41  9718.3 1240.36 10113.2 1266.37 10874.1 1281.56   10904 1282.73
#Mann= 17 ,-1 , 0
     834      .1       0  1115.5     .05       0  1287.1      .1       0
  1955.7     .16       0  2935.2      .1       0  3092.2      .1       0
    3688     .16       0  3803.8     .16       0  4148.4     .16       0
  4751.5     .05       0  5455.6     .16       0  5705.9      .1       0
  6584.2     .16       0  7060.7     .16       0    7216      .1       0
  9423.2     .16       0 10874.1      .1       0
Bank Sta=4757.9,5455.6
XS Rating Curve= 0 ,0
Exp/Cntr=0.3,0.1

Type RM Length L Ch R = 1 ,263088  ,2551,2551,2551
BEGIN DESCRIPTION:
Mapping XS a36af871
END DESCRIPTION:
XS GIS Cut Line= 4
      2901946.32     10084470.57      2901098.96     10081361.19
      2897289.25     10077720.73      2891284.54     10076813.91
#Sta/Elev= 30
  -402.8 1262.47  -218.8 1256.62   287.9 1240.52  1121.8 1229.97  1685.2 1222.84
    2060  1218.1  2668.7 1211.43    2820 1209.94  3802.4 1172.33 4494.32 1139.65
    4700 1129.28  4827.1 1117.02  5010.8 1114.51  5152.6 1126.15  5216.1 1139.88
  5371.8 1147.27  5555.8 1146.48    5865 1155.13  6404.4 1170.99  7309.8 1218.97
  7845.8 1230.92  9207.9 1248.46  9608.1 1245.03  9956.2    1253 10178.7 1251.56
 10785.3 1234.93 12186.1 1258.57   12905  1270.3 13529.4 1268.88 14162.2 1277.27
#Mann= 18 ,-1 , 0
  -402.8     .16       0  -218.8      .1       0  1121.8     .05       0
  1685.2     .05       0    2060      .1       0  2668.7      .1       0
  3802.4     .16       0 4494.32     .05       0  5216.1     .16       0
    5865      .1       0  7845.8      .1       0  9207.9     .05       0
  9608.1      .1       0  9956.2     .16       0 10785.3      .1       0
 12186.1      .1       0   12905      .1       0 13529.4      .1       0
Bank Sta=4494.32,5216.1
XS Rating Curve= 0 ,0
Exp/Cntr=0.3,0.1

Type RM Length L Ch R = 1 ,257480  ,3301,3301,3301
BEGIN DESCRIPTION:
Mapping XS 02f041a1
END DESCRIPTION:
XS GIS Cut Line= 3
      2905562.24     10082665.92      2905393.09     10078757.46
       2898203.7     10066908.27
#Sta/Elev= 30
    -923 1251.28   -48.5 1241.12   374.7 1236.21  1428.1 1218.68  2171.1 1202.14
  2984.2  1174.8  3366.6 1170.33  3621.9 1166.95    4093 1149.04  4298.5 1148.64
  4662.9 1128.65  4794.7 1111.68  5054.3  1107.4  5434.5 1133.53  6423.2 1127.66
  6496.8 1118.42  6909.1 1143.34  7057.1 1156.85  7617.6 1177.29  8018.6 1194.38
  8272.2 1195.28  9123.1  1198.3  9861.2  1200.7 10399.2 1199.45 11009.8 1225.89
 11962.4 1232.28 12565.5 1236.78 14702.8  1257.3 16356.1 1286.79 16848.8 1294.54
#Mann= 19 ,-1 , 0
    -923     .16       0   -48.5      .1       0   374.7     .16       0
  1428.1     .16       0  2171.1      .1       0  3366.6     .16       0
  3621.9      .1       0  4662.9     .05       0  5434.5     .16       0
  6909.1      .1       0  7617.6     .16       0  8272.2     .16       0
  9123.1      .1       0  9861.2      .1       0 10399.2     .16       0
 11962.4     .16       0 12565.5     .05       0 14702.8     .16       0
 16356.1     .16       0
Bank Sta=4662.9,5434.5
XS Rating Curve= 0 ,0
Exp/Cntr=0.3,0.1

Type RM Length L Ch R = 1 ,254179  ,2466,2466,2466
BEGIN DESCRIPTION:
Mapping XS a5f67f4f
END DESCRIPTION:
XS GIS Cut Line= 3
      2907468.19     10079433.95      2907972.68     10077226.52
      2901914.03     10065129.34
#Sta/Elev= 30
    10.5 1240.95   439.6 1233.49   927.4  1221.8  1258.6 1213.87    2074 1195.42
  3479.6  1139.1  4018.3  1139.6  4345.6 1142.45  4479.7 1139.21  4597.1 1127.52
    4649 1112.96  4939.5 1107.21  5821.9 1127.95  6288.4 1138.71  7064.7 1147.29
  7165.1 1142.66  7206.4 1150.75  7340.5 1146.36  7614.7 1157.15    8289 1159.21
  9075.8 1170.12  9983.8 1203.75 11548.4 1236.82 12005.9 1246.49 12297.7 1242.93
 13009.5 1240.44 13452.4 1240.98 14180.2 1240.13 15579.7 1272.34 15804.4 1277.51
#Mann= 20 ,-1 , 0
    10.5      .1       0   439.6     .05       0   927.4     .16       0
  1258.6      .1       0    2074     .08       0  4018.3     .08       0
    4649     .05       0  5821.9     .05       0  5821.9     .16       0
  6288.4     .16       0  7165.1     .05       0  7614.7     .05       0
    8289     .08       0  9075.8     .08       0 11548.4      .1       0
 12297.7     .16       0 13009.5     .16       0 13452.4     .05       0
 14180.2      .1       0 15579.7     .16       0
Bank Sta=4597.1,5821.9
XS Rating Curve= 0 ,0
Exp/Cntr=0.3,0.1

Type RM Length L Ch R = 1 ,247895  ,1553,1553,1553
BEGIN DESCRIPTION:
Mapping XS 123fdf3d
END DESCRIPTION:
XS GIS Cut Line= 3
      2910015.82     10076955.53      2913533.76     10070401.22
      2913133.41     10063419.73
#Sta/Elev= 30
   714.7  1187.7  1265.6  1181.4  2345.7 1154.08  2801.2 1142.24  3611.6  1111.5
  4131.2 1120.07  4578.3 1110.94  4580.2 1110.91  4771.9 1090.45  4979.5 1083.44
  5133.2 1097.85  5155.1 1109.78  5199.7 1125.79  5323.4 1136.08  6845.2    1124
  7240.3 1116.35  7466.6 1121.97  8361.3 1166.21  9161.9 1158.88  9493.1 1150.48
  9554.9 1157.91 10147.3 1163.38 11325.7 1174.34 12370.6  1208.3 12679.9 1220.89
 13160.8 1220.03   13457 1226.71 13781.1 1239.68 14491.3  1280.3 15146.4 1305.02
#Mann= 18 ,-1 , 0
   714.7     .05       0  1265.6     .05       0  2345.7      .1       0
  2801.2      .1       0  4580.2     .05       0  5133.2     .16       0
  5323.4     .05       0  6845.2     .05       0  7466.6      .1       0
  9161.9     .16       0  9554.9      .1       0 10147.3     .05       0
 11325.7     .16       0 12370.6     .16       0 12679.9      .1       0
 13160.8     .16       0   13457      .1       0 13781.1      .1       0
Bank Sta=4578.3,5155.1
XS Rating Curve= 0 ,0
Exp/Cntr=0.3,0.1

Type RM Length L Ch R = 1 ,246342  ,2798,2798,2798
BEGIN DESCRIPTION:
Mapping XS c0ef7d5f
END DESCRIPTION:
XS GIS Cut Line= 4
      2911378.73     10076243.07      2913197.28     10075188.92
      2913727.17     10071618.91      2914202.62     10063987.11
#Sta/Elev= 30
  1369.1 1179.16  1601.4 1187.21  1806.1 1177.63  2273.5 1161.17  2490.1 1157.38
  3033.3 1155.61  3471.9 1173.67  3790.2 1173.01  4325.5 1147.32  4511.8 1147.53
  4750.1 1140.74    4831 1117.78  4841.1 1098.79  4911.9 1079.76  5113.8 1077.93
  5624.6 1113.37  5993.8 1119.78    6883 1114.43  6964.1  1110.7  7624.1 1120.53
  7786.8 1121.78  8555.1 1154.17  8827.5 1167.81  9666.4 1164.73 10386.6 1178.92
 10822.9 1189.26 11679.7 1196.99 12645.4 1208.91 13841.7 1240.14 14726.8 1286.54
#Mann= 19 ,-1 , 0
  1369.1      .1       0  1806.1     .05       0  2273.5      .1       0
  2490.1     .05       0  3033.3      .1       0  3471.9      .1       0
  4511.8     .16       0  4841.1     .05       0  5624.6      .1       0
  5993.8     .05       0    6883      .1       0  7624.1     .05       0
  8555.1     .16       0  8827.5      .1       0  9666.4      .1       0
 10386.6      .1       0 10822.9     .16       0 11679.7     .16       0
 13841.7      .1       0
Bank Sta=4831,5624.6
XS Rating Curve= 0 ,0
Exp/Cntr=0.3,0.1

Type RM Length L Ch R = 1 ,239412  ,1931,1931,1931
BEGIN DESCRIPTION:
Mapping XS c23ee2bb
END DESCRIPTION:
XS GIS Cut Line= 3
      2915306.55     10075909.28      2916966.84     10073603.15
      2919507.66     10073113.46
#Sta/Elev= 30
  1282.5 1168.29  1410.3 1168.51    1707 1151.82  2131.1 1135.32  2324.7 1127.29
  2526.5 1120.37  2893.3 1108.96  2920.1 1108.53  3174.7 1105.21  3809.7 1104.39
  3931.2 1100.73  4421.1 1109.35  4635.9 1101.77  4685.9 1098.88  4828.5  1083.1
    4859  1074.8  5113.4 1073.62  5174.7  1081.7    5246 1078.53  5429.3 1083.01
  5612.6 1097.89  5622.4 1099.54  5704.3 1112.32  5826.5 1117.62  6000.8 1147.41
  6040.4  1144.6  6099.5 1155.32  6459.7 1180.07    6561 1176.39  6711.7 1168.46
#Mann= 13 ,-1 , 0
  1282.5      .1       0    1707     .05       0  2131.1      .1       0
  2324.7     .05       0  2526.5      .1       0  2893.3     .05       0
  2920.1      .1       0  3174.7     .05       0  4635.9      .1       0
  4685.9     .05       0  5622.4      .1       0  6459.7     .05       0
    6561      .1       0
Bank Sta=4685.9,5612.6
XS Rating Curve= 0 ,0
Exp/Cntr=0.3,0.1

Type RM Length L Ch R = 1 ,237481  ,1337,1337,1337
BEGIN DESCRIPTION:
Mapping XS cc62e269
END DESCRIPTION:
XS GIS Cut Line= 3
      2915686.76     10076052.81       2919837.8     10074506.45
      2920265.51     10073608.86
#Sta/Elev= 30
  2850.6 1152.82  2945.7 1151.93    3092 1156.95  3202.6 1155.07  3348.9 1140.71
  3739.9 1118.97  3919.5 1116.31  4271.1 1105.08  4446.3 1103.33  4665.7 1103.83
  4681.5 1104.65  4772.7 1104.98  4810.4  1103.5  4840.7 1097.58    4848 1093.34
  4896.1 1074.87  4965.1 1060.22    5012 1063.31  5061.4 1074.19  5104.1 1076.62
  5221.5 1066.27  5317.5 1066.41  5495.6  1083.7    5642 1085.23  5702.6 1091.32
  5838.3 1099.48  7098.1 1149.94  7550.9 1154.79    7690 1156.18  8274.6 1165.59
#Mann= 13 ,-1 , 0
  2850.6      .1       0  3739.9     .05       0  3919.5     .05       0
  4271.1      .1       0  4446.3     .05       0  4665.7     .16       0
  4681.5      .1       0  4772.7     .16       0  4840.7     .05       0
  5702.6     .16       0  7550.9     .05       0  7550.9     .16       0
    7690     .05       0
Bank Sta=4848,5702.6
XS Rating Curve= 0 ,0
Exp/Cntr=0.3,0.1

Type RM Length L Ch R = 1 ,233047  ,2127,2127,2127
BEGIN DESCRIPTION:
Mapping XS 1c776ee1
END DESCRIPTION:
XS GIS Cut Line= 3
       2913276.2     10076999.55      2916235.35     10078142.64
      2918494.15     10079710.73
#Sta/Elev= 30
  1169.8 1135.37  1445.3 1124.73  1638.9 1108.26    1987 1090.01  2443.3 1114.65
  2789.4 1103.32  2904.9 1097.27  3037.5 1098.16  3344.2 1100.66  3779.4 1083.66
  4136.7 1088.52    4561 1072.68  4820.1 1055.54  5279.6 1059.17  5330.3  1065.7
  5336.4 1074.22  5357.3 1086.44    5387 1090.91  5422.8 1105.44  5530.2 1122.59
  5631.5  1123.7  6090.8 1147.99    6200 1146.14  6228.1 1144.89  6350.1 1144.89
  6476.4 1158.95  6514.2 1169.19  6609.6 1173.75  7031.5 1175.26  7091.8 1174.91
#Mann= 12 ,-1 , 0
  1169.8      .1       0  2789.4     .05       0  2904.9      .1       0
  3037.5     .16       0  3344.2      .1       0    4561     .05       0
  5336.4     .05       0    6200      .1       0  6228.1     .05       0
  6476.4      .1       0  6609.6     .05       0  7031.5      .1       0
Bank Sta=4561,5336.4
XS Rating Curve= 0 ,0
Exp/Cntr=0.3,0.1

Type RM Length L Ch R = 1 ,230920  ,1173,1173,1173
BEGIN DESCRIPTION:
Mapping XS 7631730a
END DESCRIPTION:
XS GIS Cut Line= 3
      2912207.63     10077420.49      2915847.58     10079678.72
      2917472.07     10079937.36
#Sta/Elev= 30
  2033.1 1135.37  2275.8 1125.83  2507.3 1100.19  2595.9 1109.75  2711.7 1112.71
  3110.9 1082.25  3191.7 1088.88  3373.2 1086.82  3715.6 1091.98  3961.7  1079.8
  4308.6 1074.41  4366.5 1069.98  4411.3 1059.61    4480 1074.85    4513 1076.41
  4549.6 1070.94  4555.5 1069.02  4707.8 1054.65  5021.8 1051.99  5159.1 1056.12
  5232.3 1071.81  5411.8 1109.48  5542.9    1128    5863 1156.37  6183.1 1168.04
  6631.6 1157.79  6854.2 1157.76  6946.4  1167.4  7842.3 1204.55  7961.6 1202.05
#Mann= 9 ,-1 , 0
  2033.1      .1       0  3191.7     .05       0  3715.6      .1       0
  3961.7     .05       0    4480     .16       0  4555.5     .05       0
  5232.3      .1       0  6631.6     .05       0  6946.4      .1       0
Bank Sta=4549.6,5232.3
XS Rating Curve= 0 ,0
Exp/Cntr=0.3,0.1

Type RM Length L Ch R = 1 ,229747  ,1902,1902,1902
BEGIN DESCRIPTION:
Mapping XS e6b95da8
END DESCRIPTION:
XS GIS Cut Line= 4
      2909507.91      10078837.1      2910952.38     10078609.97
      2914994.68     10080210.81      2917033.67     10080279.21
#Sta/Elev= 30
   411.7 1196.17   654.4 1194.31   846.6  1182.3  1195.9 1166.04  1820.9 1155.48
  2137.7 1130.69  2737.6 1117.57  3283.1 1089.11  3317.9 1087.16  3422.3 1084.39
    3578 1078.12  3661.8 1064.56  3691.5  1067.9  3965.2 1063.46  4067.6 1062.59
  4261.5 1070.56  4464.4  1077.3    4480 1077.67  4526.3 1075.47  4537.3 1074.09
  4645.4 1057.05  4762.7 1050.17  5139.4 1052.81  5377.8 1074.08  6112.6 1104.55
  6114.8 1104.61  6454.3 1108.05  6955.9 1134.72    7206 1164.23  8261.8 1193.68
#Mann= 15 ,-1 , 0
   411.7      .1       0   846.6     .05       0  1195.9      .1       0
  3283.1     .05       0  3317.9     .16       0  3422.3      .1       0
  3965.2     .05       0  4067.6      .1       0  4261.5     .05       0
  4464.4      .1       0    4480     .05       0  4526.3     .05       0
  5377.8      .1       0  6112.6     .05       0  6114.8      .1       0
Bank Sta=4537.3,5377.8
XS Rating Curve= 0 ,0
Exp/Cntr=0.3,0.1

Type RM Length L Ch R = 1 ,227845  ,1435,1435,1435
BEGIN DESCRIPTION:
Mapping XS ffaed9bf
END DESCRIPTION:
XS GIS Cut Line= 3
      2909730.33     10083353.82      2910877.68     10082433.77
      2917051.75     10080583.28
#Sta/Elev= 30
   444.9 1194.25   752.1 1197.66   901.4 1202.16    1200    1195  1675.5 1187.92
  1908.9 1179.85  2485.8 1142.68  2676.4 1129.03  2735.1 1125.01  2877.2 1130.63
  3565.4 1119.12  4064.2 1097.15  4301.7 1087.59  4576.8 1095.24  4686.4 1088.28
  4752.6 1076.88 4760.42 1067.18  4776.8 1047.45  4785.7 1046.07  5065.7 1045.16
  5520.7 1066.37  5875.1 1083.88  6500.5 1108.33  6874.5 1114.38  7076.6 1124.56
  7230.9 1135.77    7512 1166.86  7735.7 1168.88  7820.8 1168.58    8361 1193.22
#Mann= 19 ,-1 , 0
   444.9      .1       0   752.1     .05       0   901.4      .1       0
    1200     .16       0  1675.5      .1       0  2485.8     .05       0
  2676.4      .1       0  2877.2     .16       0  4064.2      .1       0
  4752.6     .05       0  5520.7     .05       0  5520.7      .1       0
  5520.7     .16       0  5875.1      .1       0  6500.5     .16       0
  7076.6      .1       0  7230.9     .16       0  7735.7      .1       0
  7820.8     .16       0
Bank Sta=4760.42,5520.7
XS Rating Curve= 0 ,0
Exp/Cntr=0.3,0.1

Type RM Length L Ch R = 1 ,226410  ,1844,1844,1844
BEGIN DESCRIPTION:
Mapping XS 5c696f8a
END DESCRIPTION:
XS GIS Cut Line= 3
      2910330.36     10083691.03      2913498.94     10083542.37
      2917051.49     10080960.88
#Sta/Elev= 30
   233.7 1214.73   372.5 1209.62   982.6  1185.1  1312.9 1181.97  1573.3 1180.89
  2200.1 1159.44  2832.5 1123.48  3006.5 1113.18  3239.6 1103.28  3353.8 1097.89
  3494.3 1093.01  3716.2 1086.88  4140.7 1066.58  4399.5 1064.33  4535.5  1071.1
  4667.4 1063.09  4707.1 1054.99  4736.4 1044.35  4972.7 1041.83  5194.8  1043.3
  5330.8 1053.67    5337 1054.83    5732 1077.55    6036 1090.48  6161.9 1095.15
    6305 1099.49  6990.2 1113.38  7105.4 1124.38    7321 1164.84  7797.2 1183.88
#Mann= 18 ,-1 , 0
   233.7     .16       0   372.5      .1       0  1312.9     .16       0
  2200.1      .1       0  2832.5     .05       0  3006.5      .1       0
  3239.6     .05       0  3353.8      .1       0  3494.3     .05       0
  3716.2      .1       0  4399.5     .16       0  4667.4      .1       0
  4707.1     .05       0    5337     .16       0    5732      .1       0
    6036     .16       0  6161.9      .1       0    6305     .16       0
Bank Sta=4707.1,5330.8
XS Rating Curve= 0 ,0
Exp/Cntr=0.3,0.1

Type RM Length L Ch R = 1 ,224566  ,1351,1351,1351
BEGIN DESCRIPTION:
Mapping XS da71cbba
END DESCRIPTION:
XS GIS Cut Line= 3
      2914057.84     10087236.76      2916050.38     10084448.67
      2917235.64     10081234.01
#Sta/Elev= 30
   482.2 1179.64   584.9 1183.88   912.8 1157.98  1018.9 1149.85    1382 1134.85
  1498.6 1130.03  2047.2 1112.59  2203.2 1109.34  2437.8 1104.34    2907 1112.68
  3087.2  1116.6  3190.3 1124.21  3573.8 1153.98  3845.1 1149.52  4023.2 1138.24
  4287.4 1102.19  4489.9  1058.4  4495.7 1055.93  4637.2 1038.96  5102.7 1032.85
    5236 1034.71  5330.5 1051.09  5335.8 1053.69  5421.8 1062.92  5515.4 1064.01
  5737.7  1067.6  6494.8 1104.35  6747.5    1132  6869.2 1133.92  7335.3 1171.32
#Mann= 17 ,-1 , 0
   482.2      .1       0   584.9     .16       0   912.8     .05       0
  1018.9      .1       0    1382     .16       0  1498.6      .1       0
  2047.2      .1       0  2203.2     .16       0  2437.8     .05       0
    2907     .16       0  3190.3      .1       0  3845.1     .16       0
  4023.2      .1       0  4489.9     .05       0  5330.5     .16       0
  5515.4      .1       0  5737.7     .16       0
Bank Sta=4495.7,5335.8
XS Rating Curve= 0 ,0
Exp/Cntr=0.3,0.1

Type RM Length L Ch R = 1 ,223215  ,1370,1370,1370
BEGIN DESCRIPTION:
Mapping XS 223380d4
END DESCRIPTION:
XS GIS Cut Line= 3
      2916039.69     10088719.39      2918178.79     10082474.73
      2918002.84     10081557.32
#Sta/Elev= 30
  -202.3 1208.22   -14.8 1196.84   738.5 1149.07   881.9 1143.72  1040.4 1155.71
  1227.1 1161.68  1602.5 1190.08  2003.9 1184.66  2177.9 1172.15  2337.5 1154.82
  2694.3 1157.83  2963.3 1138.86  3206.5 1112.29  3372.4 1103.74  3514.5 1098.19
  3713.5 1089.17  4292.6 1062.56  4532.3 1048.17  4714.7 1031.95  5115.9 1030.27
  5226.3 1033.51  5267.3 1047.04  5272.6 1049.06  5310.9 1064.61  5543.4 1081.25
  5678.7 1089.15  6044.1 1109.87  6425.9 1154.87  7117.2 1163.92  7332.7 1173.09
#Mann= 16 ,-1 , 0
  -202.3     .05       0   -14.8     .05       0   738.5      .1       0
  1040.4      .1       0  2177.9      .1       0  2694.3     .16       0
  2963.3      .1       0  3206.5      .1       0  3372.4     .05       0
  3514.5      .1       0  3713.5     .05       0  4292.6     .05       0
  4532.3     .05       0  5267.3     .05       0  5543.4      .1       0
  5678.7     .16       0
Bank Sta=4532.3,5272.6
XS Rating Curve= 0 ,0
Exp/Cntr=0.3,0.1

Type RM Length L Ch R = 1 ,221845  ,1447,1447,1447
BEGIN DESCRIPTION:
Mapping XS c9dd96ed
END DESCRIPTION:
XS GIS Cut Line= 3
      2918283.86     10087496.93      2919231.19     10083300.16
      2919054.57     10080714.64
#Sta/Elev= 30
  1683.1 1214.09  1843.4 1202.58  2078.3 1179.46  2631.2 1130.37  2651.7 1128.26
  3019.1 1103.98  3190.1 1106.74  3997.8 1114.14    4116 1104.35    4321  1071.4
  4442.6 1058.32  4585.2 1043.75  4816.6 1028.74  5099.9 1026.11  5171.9 1028.77
  5220.9 1045.06  5226.9 1046.36  5243.7 1054.05  5312.4 1066.07    5704 1085.64
  6122.2 1112.49  6535.3 1118.29  6625.3 1117.66  6964.4 1107.44  7104.1 1102.07
  7419.8  1113.8  7495.4 1109.73    7766  1133.5    8301  1151.6    8577 1168.72
#Mann= 14 ,-1 , 0
  1683.1      .1       0  1843.4     .16       0  2078.3      .1       0
  2631.2     .16       0  2651.7      .1       0  3190.1     .16       0
  4442.6      .1       0  4585.2     .05       0  5226.9     .16       0
    5704      .1       0  6535.3     .05       0  6625.3      .1       0
  6964.4     .05       0  7104.1      .1       0
Bank Sta=4585.2,5220.9
XS Rating Curve= 0 ,0
Exp/Cntr=0.3,0.1

Type RM Length L Ch R = 1 ,209613  ,1569,1569,1569
BEGIN DESCRIPTION:
Mapping XS c5e8d5e5
END DESCRIPTION:
XS GIS Cut Line= 2
      2928327.79     10077777.99      2921856.64     10077115.21
#Sta/Elev= 30
  2503.5 1121.47  2610.5 1120.19  2814.4 1121.04  3016.3 1114.15  3192.2 1091.49
  3548.3 1056.16  3706.8  1065.1  3901.1 1076.94  4410.7 1075.11  4583.6 1058.13
  4633.9 1047.58  4664.1 1027.65  4694.2  1018.9  4865.1 1010.84  4905.3 1002.32
    4950 1001.42    5418  1011.2  5528.6 1026.49  5536.2 1027.17  5850.4 1028.47
  6306.2 1042.66  6936.8 1068.14  7158.7 1076.57  7363.1 1069.98  7628.1 1087.05
  7781.8 1097.06  8220.7 1123.97  8466.5 1142.97    8912  1159.2  9008.5 1158.38
#Mann= 19 ,-1 , 0
  2503.5      .1       0  2610.5      .1       0  3016.3     .16       0
  3192.2      .1       0  3706.8     .05       0  3901.1      .1       0
  4410.7     .16       0  4664.1     .05       0  5536.2      .1       0
  5850.4      .1       0  6306.2     .05       0  6936.8      .1       0
  7158.7     .16       0  7363.1      .1       0  7628.1     .05       0
  7781.8      .1       0  8220.7     .05       0  8466.5      .1       0
    8912      .1       0
Bank Sta=4664.1,5528.6
XS Rating Curve= 0 ,0
Exp/Cntr=0.3,0.1
