HEC-RAS study PEDERNALES RIVER.prj: PEDERNALES RIVER Base Level Engineering

--- PEDERNALES RIVER.g02 (geometry) --- (continued)

Type RM Length L Ch R = 1 ,107762  ,2052,2052,2052
BEGIN DESCRIPTION:
PEDERNALES RIVER 291.0
END DESCRIPTION:
XS GIS Cut Line= 2
      2970090.64     10100965.07      2972552.92     10091360.05
#Sta/Elev= 30
  1435.6 1039.93  1552.1 1035.28  1987.5 1020.37  2451.8 1024.49  2895.1 1010.38
  3299.9  978.93    3391  952.13  3630.6  920.98  4482.4  878.09  4657.9  831.28
  4688.8  801.42  4788.1  752.23  4946.1  722.68  5032.6  721.43  5272.4  768.03
    5675  802.92  5680.2  804.17  6072.2  833.17  6317.2  870.56  6970.8  880.98
  7573.4  887.78  8159.5  894.88  8578.4  898.91  9581.9  908.36  9936.3  914.47
 10647.5  929.68 10873.9  970.74 11025.4   973.5 11344.9  972.29 11351.2  972.15
#Mann= 18 ,-1 , 0
  1435.6      .1       0  1552.1     .16       0  1987.5     .16       0
  2451.8      .1       0  2895.1     .16       0    3391      .1       0
  3630.6     .16       0  4688.8    .035       0    5675     .16       0
  6970.8     .05       0  7573.4     .16       0  8159.5      .1       0
  8578.4     .16       0  9581.9     .16       0  9936.3     .05       0
 10647.5     .16       0 11025.4      .1       0 11344.9     .16       0
Bank Sta=4688.8,5680.2
XS Rating Curve= 0 ,0
Exp/Cntr=0.3,0.1

Type RM Length L Ch R = 1 ,105710  ,1972,1972,1972
BEGIN DESCRIPTION:
PEDERNALES RIVER 292.0
END DESCRIPTION:
XS GIS Cut Line= 3
      2972195.43     10099365.22      2972991.31     10098181.44
      2972638.06     10091646.83
#Sta/Elev= 30
  2550.7 1054.36    2601 1054.68  2659.5 1054.79  2957.8 1035.84    3179  987.42
    3396  931.26  4071.4  883.75  4265.3  870.15  4545.7  808.57  4585.7  788.72
  4625.8  789.18  4665.9  765.92    4936  718.82  5126.5  731.95  5196.6  755.35
  5246.7  795.52  5256.7  804.04    5457  858.25  5608.3  868.25  6438.4  878.79
  7191.2  865.05  8009.3  881.61  8049.2  882.58  8272.1  887.98  9461.4  901.04
  9658.8  906.74  9757.5  908.64 10169.6  931.02   10418  972.39 10521.3  975.42
#Mann= 16 ,-1 , 0
  2550.7      .1       0    2601     .05       0  2659.5      .1       0
    3179     .05       0  4071.4     .16       0  4545.7    .035       0
  5246.7     .16       0  7191.2      .1       0  8009.3     .16       0
  8049.2      .1       0  8272.1     .16       0  9461.4     .05       0
  9658.8     .16       0  9757.5      .1       0 10169.6     .16       0
   10418      .1       0
Bank Sta=4545.7,5256.7
XS Rating Curve= 0 ,0
Exp/Cntr=0.3,0.1

Type RM Length L Ch R = 1 ,103738  ,2199,2199,2199
BEGIN DESCRIPTION:
PEDERNALES RIVER 293.0
END DESCRIPTION:
XS GIS Cut Line= 3
      2976670.08     10097271.99      2973330.17     10095342.73
      2972791.98     10091496.78
#Sta/Elev= 30
  2054.5 1011.85  2391.3  1010.6  2581.3  988.73  2927.1  979.66  3282.4  926.58
  3397.8  911.22  3631.5  897.21  4564.1  864.22  4595.7  835.87  4712.5  800.99
  4740.7  788.98  4756.5   759.5  4799.6  738.83  4885.7  718.34  4989.4  715.21
  5209.1  746.42  5421.2  800.84  5428.5  802.33  5786.5  855.39    5839  848.53
  5909.7  861.93  6122.6  858.96  6274.1  816.26  6486.1  856.45  7021.3  880.59
  8487.9  887.29  8637.1  896.24  8819.1  901.68  9528.5  935.14    9795  956.63
#Mann= 11 ,-1 , 0
  2054.5     .16       0  2927.1      .1       0  3282.4     .05       0
  3397.8      .1       0  3631.5     .16       0  4712.5    .035       0
  5428.5     .16       0  8487.9      .1       0  8637.1     .16       0
  8819.1      .1       0  9528.5     .16       0
Bank Sta=4712.5,5421.2
XS Rating Curve= 0 ,0
Exp/Cntr=0.3,0.1

Type RM Length L Ch R = 1 ,101539  ,2438,2438,2438
BEGIN DESCRIPTION:
PEDERNALES RIVER 294.0
END DESCRIPTION:
XS GIS Cut Line= 4
      2978220.18     10095759.74      2973306.44     10092986.37
      2973046.06     10091225.33      2972471.27     10090328.59
#Sta/Elev= 30
   680.3 1004.91   706.3 1004.35  1177.5  981.49  1704.8  941.17    1921  948.26
  2294.4  927.57  2537.5  917.02  2783.7  906.34  3103.3  892.47  3251.7  886.03
  3640.5  867.45  4115.3  854.47  4253.4  826.26  4671.2  799.15  4678.3  795.74
  4811.4  734.83  5032.1  712.55  5199.8  752.89  5264.8  796.69  5501.7  866.81
  5686.3  870.19  6239.7  867.88    6503  875.45  6983.4  890.03    7143  894.87
  8082.8   911.4    8439  910.11  8935.9  930.45  9050.9  965.76    9168  969.35
#Mann= 19 ,-1 , 0
   680.3     .16       0   706.3      .1       0  1177.5     .16       0
    1921      .1       0  2294.4     .16       0  2537.5     .05       0
  2783.7      .1       0  3103.3     .16       0  3251.7     .05       0
  3640.5     .16       0  4671.2    .035       0  5264.8     .16       0
  5686.3     .16       0  6239.7      .1       0    6503     .16       0
  6983.4     .16       0    7143      .1       0  8082.8     .05       0
    8439     .16       0
Bank Sta=4678.3,5264.8
XS Rating Curve= 0 ,0
Exp/Cntr=0.3,0.1

Type RM Length L Ch R = 1 ,99101   ,1723,1723,1723
BEGIN DESCRIPTION:
PEDERNALES RIVER 295.0
END DESCRIPTION:
XS GIS Cut Line= 3
      2978986.28     10095226.64      2976638.87     10092007.54
      2972412.01     10089959.45
#Sta/Elev= 30
  -244.2  1013.2    64.3     986   587.3  962.04  1169.5  910.05  1380.6  898.43
  2258.8  887.23  2475.1  888.95  2761.8   899.1  2890.1  900.51  4395.9  847.49
  4565.5  818.21  4700.9  793.81  4873.8  714.24  5067.5  710.21  5218.2  752.65
  5373.8  812.92  5383.9  816.53  5530.4  852.75  6060.6  868.37  6262.5  868.77
  6500.5   870.6  6778.1  872.22  7003.7  865.34  7497.8  893.33  7672.3  901.87
  7817.5   911.9  7994.7  926.79  8182.9  964.46  8346.5  963.81  8436.8  950.89
#Mann= 18 ,-1 , 0
  -244.2     .16       0  1169.5     .05       0  1380.6     .05       0
  2258.8      .1       0  2475.1     .05       0  2761.8     .05       0
  2890.1     .16       0  4565.5    .033       0  5373.8     .16       0
  6060.6      .1       0  6262.5     .16       0  6500.5     .16       0
  6778.1      .1       0  7003.7     .16       0  7497.8     .05       0
  7672.3      .1       0  7817.5     .16       0  7994.7     .16       0
Bank Sta=4565.5,5383.9
XS Rating Curve= 0 ,0
Exp/Cntr=0.3,0.1

Type RM Length L Ch R = 1 ,97378   ,1923,1923,1923
BEGIN DESCRIPTION:
PEDERNALES RIVER 296.0
END DESCRIPTION:
XS GIS Cut Line= 3
      2979228.19     10094969.25      2977394.83     10090541.16
      2972783.04       10087989.
#Sta/Elev= 30
  -869.8  997.71  -366.1  940.26   209.7  935.28   367.9  907.96  1183.5  874.29
  1717.3  852.59  1938.2  851.05  2388.9  859.35  2892.2  872.67  3112.6  870.69
  3486.7  865.63  4212.6  847.58  4462.3   837.1  4593.7  809.81  4778.1  745.21
  4831.9  746.12    4947  705.58    5073  706.83  5331.2  796.35  5427.3  811.94
  5537.3  840.76  5873.5   846.3  6400.4  858.39  6620.5     864  7168.7  877.96
  7849.1  895.29  8385.3  908.95  8534.5  933.18  8634.9  956.93  9193.7  960.98
#Mann= 19 ,-1 , 0
  -869.8     .16       0   209.7     .05       0  1183.5      .1       0
  1717.3     .05       0  1938.2      .1       0  2388.9     .05       0
  2892.2     .16       0  3112.6     .05       0  3486.7      .1       0
  4212.6     .05       0  4462.3     .16       0  4593.7    .033       0
  5427.3     .16       0  5873.5     .16       0  6400.4     .05       0
  6620.5     .16       0  7168.7      .1       0  7849.1      .1       0
  8534.5     .16       0
Bank Sta=4593.7,5427.3
XS Rating Curve= 0 ,0
Exp/Cntr=0.3,0.1

Type RM Length L Ch R = 1 ,95455   ,2491,2491,2491
BEGIN DESCRIPTION:
PEDERNALES RIVER 297.0
END DESCRIPTION:
XS GIS Cut Line= 3
       2979593.3     10095277.54      2977765.04     10090437.22
      2979397.27     10086551.07
#Sta/Elev= 30
  -896.6  997.42  -865.9  995.48  -234.7  964.58     513     918   735.9  902.86
  1901.6  856.32  2372.1  842.49  2639.6  841.85  3063.1  846.31  3474.2  850.64
  3848.9  854.59  4461.7  845.53  4617.5  810.12  4628.4  803.59  4877.8  709.94
  4975.5  701.44    5100  714.51  5406.8  808.61  5420.1  815.06  5435.9  848.14
  5459.7  858.45  5724.4  880.47  6054.9  952.96  6257.7  959.62  6733.1  964.55
  6991.1  959.09  7339.9  917.05  7702.9  959.85  8268.8  983.06  8492.5  984.56
#Mann= 19 ,-1 , 0
  -896.6     .16       0  -865.9      .1       0  -234.7     .16       0
     513      .1       0   735.9     .05       0  1901.6     .05       0
  2372.1     .16       0  2639.6     .05       0  3063.1      .1       0
  3474.2      .1       0  3848.9      .1       0  4461.7      .1       0
  4617.5    .035       0  5420.1     .16       0  6257.7      .1       0
  6733.1     .16       0  6991.1     .16       0  7702.9      .1       0
  8268.8      .1       0
Bank Sta=4628.4,5406.8
XS Rating Curve= 0 ,0
Exp/Cntr=0.3,0.1

Type RM Length L Ch R = 1 ,92964   ,1831,1831,1831
BEGIN DESCRIPTION:
PEDERNALES RIVER 298.0
END DESCRIPTION:
XS GIS Cut Line= 3
      2979808.14     10095453.83      2979738.51     10092306.24
      2981802.31     10086862.91
#Sta/Elev= 30
   265.2 1000.22     650  978.98  1575.6  947.36  2077.2  904.52  2420.9  879.03
  2906.3   864.7  3143.9  862.52  3429.3  860.28  3661.5  854.91  3954.3  848.14
  4512.1  837.11  4615.8  821.21  4646.1  795.94  4810.8  752.15  4865.7     716
  5035.7  698.89  5266.4  772.13  5346.1  781.33  5416.1  820.83  5632.9  837.73
  6465.6   852.7  6779.6  863.92  7159.4  935.48  7517.6   935.5  7855.9  905.59
  8143.4   930.7  8319.4  928.91  8764.6  990.54  9220.5 1045.56    9235 1048.43
#Mann= 19 ,-1 , 0
   265.2     .16       0     650     .16       0  2077.2     .16       0
  2420.9     .05       0  2906.3      .1       0  3143.9     .05       0
  3429.3     .16       0  3661.5     .05       0  3954.3      .1       0
  4512.1     .16       0  4615.8    .035       0  5416.1     .16       0
  5632.9      .1       0  6465.6     .05       0  6779.6     .16       0
  7855.9     .16       0  8319.4      .1       0  8764.6      .1       0
  9220.5      .1       0
Bank Sta=4615.8,5416.1
XS Rating Curve= 0 ,0
Exp/Cntr=0.3,0.1

Type RM Length L Ch R = 1 ,91133   ,1601,1601,1601
BEGIN DESCRIPTION:
PEDERNALES RIVER 299.0
END DESCRIPTION:
XS GIS Cut Line= 3
      2979956.55     10095737.77      2981713.59     10092287.23
      2983577.82     10087188.69
#Sta/Elev= 30
   290.9 1006.08  1021.1  979.74  1356.9  966.97  1441.3  964.25  1519.5  961.83
  1991.1  942.83  2221.8  933.86  2468.4  906.61  2705.6  891.69  2745.3  890.25
  2853.3  886.33  2942.8  883.08  4562.7  828.07  4645.9   811.9  4677.8  785.19
    4684  781.61  4954.7  700.51  5096.2  699.18  5324.7  786.41    5338  787.65
  5369.9   791.7  5380.5  810.75  5416.3  798.61  5472.1  819.35  6608.7  848.87
  6667.5  848.94  7310.4  854.33  7452.4  877.54  8620.4  907.66  9591.7 1003.94
#Mann= 17 ,-1 , 0
   290.9     .16       0  1021.1      .1       0  1356.9     .16       0
  1441.3      .1       0  1519.5     .16       0  1991.1      .1       0
  2221.8      .1       0  2468.4     .05       0  2705.6      .1       0
  2745.3     .05       0  2853.3      .1       0  2942.8     .16       0
  4562.7     .05       0    4684    .035       0    5338     .16       0
  6608.7      .1       0  6667.5     .16       0
Bank Sta=4677.8,5324.7
XS Rating Curve= 0 ,0
Exp/Cntr=0.3,0.1

Type RM Length L Ch R = 1 ,89532   ,1871,1871,1871
BEGIN DESCRIPTION:
PEDERNALES RIVER 300.0
END DESCRIPTION:
XS GIS Cut Line= 3
      2980085.16     10095869.54      2983134.42     10093216.25
       2984647.2     10088460.59
#Sta/Elev= 30
  -292.9  1007.9  -171.7  999.78   514.6  954.15  1301.7   957.5  1846.7  898.03
  2168.5   899.7  2279.5  895.97  2435.8   882.4  2608.1  869.04  2910.2  854.54
  3076.1   853.8  4508.6  837.29  4654.2  823.65  4675.2  789.13  4707.3  785.54
  4964.9  698.64    5074  700.31  5315.3  784.06  5336.3  810.85  6024.6  852.76
  6163.7  861.21  6367.4  886.07  6844.2  936.74  7139.9  930.64  7487.5  981.41
  7985.3  997.76    8302 1009.36  8505.7 1024.69  8607.5 1028.88  8739.6 1025.98
#Mann= 18 ,-1 , 0
  -292.9      .1       0  -171.7     .16       0  2168.5      .1       0
  2279.5      .1       0  2435.8     .16       0  2608.1     .05       0
  2910.2     .16       0  3076.1     .16       0  4707.3    .035       0
  5315.3     .16       0  6024.6     .16       0  6163.7      .1       0
  6367.4     .16       0  6844.2      .1       0  7985.3     .16       0
    8302      .1       0  8505.7     .16       0  8607.5      .1       0
Bank Sta=4707.3,5315.3
XS Rating Curve= 0 ,0
Exp/Cntr=0.3,0.1

Type RM Length L Ch R = 1 ,87661   ,2509,2509,2509
BEGIN DESCRIPTION:
PEDERNALES RIVER 320.0
END DESCRIPTION:
XS GIS Cut Line= 4
      2981795.05      10095316.6      2985357.45     10093641.85
      2985422.46     10088382.18       2984808.8     10087463.12
#Sta/Elev= 30
  -446.8  967.96   421.1   933.3  1347.1  940.02  2203.7   887.7  2689.2  865.38
  3084.1  858.53  3296.2  858.46  3498.3  856.17    4088  828.75  4284.6  820.87
  4647.8  814.34  4667.8  784.07  4967.6  699.65  5067.9  701.26  5277.9  782.83
  5297.9  810.33  5464.1  818.44  5856.3  831.71  6193.1  841.21    6447   848.2
  6643.6  854.87    7445  862.13  7823.1  894.52  8438.1  921.48  8688.1  868.81
    8844  925.44  9270.5  979.21  9549.4  989.02    9761 1005.88  9854.8 1017.41
#Mann= 19 ,-1 , 0
  -446.8     .16       0  2203.7     .05       0  2689.2     .16       0
  3084.1     .05       0  3296.2     .16       0  3498.3     .16       0
    4088     .05       0  4284.6     .16       0  4667.8    .033       0
  5277.9     .16       0  5464.1      .1       0  5856.3     .05       0
  6193.1      .1       0    6447     .05       0  6643.6     .16       0
    7445      .1       0  7823.1     .16       0  9549.4      .1       0
    9761     .16       0
Bank Sta=4667.8,5277.9
XS Rating Curve= 0 ,0
Exp/Cntr=0.3,0.1

Type RM Length L Ch R = 1 ,85152   ,3600,3600,3600
BEGIN DESCRIPTION:
PEDERNALES RIVER 301.0
END DESCRIPTION:
XS GIS Cut Line= 3
      2980915.77     10096577.44      2987819.33     10092864.99
      2988107.51     10087108.96
#Sta/Elev= 30
   -3847   968.9 -2844.8  898.07 -1923.9  930.25   198.2  907.36   564.3  873.34
  1659.1  839.32    2207  872.11  2403.5  895.58  2814.5  867.72  3043.8  854.01
  3273.1  841.81  3502.4   835.5  3974.1   821.6  4161.7  814.56  4431.6   804.2
  4613.5  797.21  4653.5  772.59  4663.6  768.37  4883.6  697.66  5084.1  699.57
  5304.4  774.16  5334.4  800.29  5496.8   814.1  5667.4  823.58  5871.1   834.9
  6264.1  856.74  6460.6  867.65  6755.4  912.49  8137.9 1004.93  9754.7 1025.31
#Mann= 19 ,-1 , 0
   -3847     .16       0   564.3     .16       0    2207      .1       0
  2403.5     .16       0  2814.5     .16       0  3043.8     .05       0
  3273.1     .05       0  3502.4     .16       0  3974.1     .05       0
  4161.7     .05       0  4431.6     .16       0  4653.5    .033       0
  5304.4     .16       0  5496.8      .1       0  5667.4     .05       0
  5871.1     .16       0  6264.1     .05       0  6460.6      .1       0
  6755.4     .16       0
Bank Sta=4663.6,5304.4
XS Rating Curve= 0 ,0
Exp/Cntr=0.3,0.1

Type RM Length L Ch R = 1 ,81552   ,1601,1601,1601
BEGIN DESCRIPTION:
PEDERNALES RIVER 302.0
END DESCRIPTION:
XS GIS Cut Line= 4
      2982870.73     10099240.47      2987246.08     10094997.67
      2990718.78     10094259.36        2990581.     10088554.41
#Sta/Elev= 30
 -2730.4  956.69 -1816.2  928.95  -599.4  894.28  -222.3  909.15  1367.3  881.57
  1761.7   879.3  2425.6  859.36  4179.3  824.19  4736.7  808.65  4767.3  781.68
  4777.6  771.28  4971.6   685.3  5166.1   698.6  5442.1  772.82  5462.5  784.31
  5570.5     825  6028.6  857.83  6244.5  900.19  6531.9   877.1  7010.8  882.89
  7504.5  946.18  8636.7   981.3  9087.4  975.95  9481.3  968.28 10071.1   979.9
   10738  952.85 11316.9  977.29 12111.3 1043.19 12488.1  1061.1 12621.2 1062.16
#Mann= 20 ,-1 , 0
 -2730.4     .05       0 -1816.2      .1       0  -599.4      .1       0
  -222.3     .16       0  1367.3     .16       0  1761.7     .16       0
  2425.6     .05       0  4179.3     .16       0  4777.6    .035       0
  5442.1      .1       0  6028.6      .1       0  7010.8     .16       0
  7504.5      .1       0  8636.7     .05       0  9087.4     .16       0
  9481.3      .1       0   10738     .16       0 11316.9     .16       0
 12111.3     .16       0 12488.1      .1       0
Bank Sta=4767.3,5462.5
XS Rating Curve= 0 ,0
Exp/Cntr=0.3,0.1

Type RM Length L Ch R = 1 ,79951   ,2522,2522,2522
BEGIN DESCRIPTION:
PEDERNALES RIVER 303.0
END DESCRIPTION:
XS GIS Cut Line= 4
      2983075.13     10099555.52      2987168.58     10097054.02
      2991987.23     10094874.01      2990994.39     10088819.99
#Sta/Elev= 30
 -1802.4  968.12 -1745.4  966.68 -1026.6  905.72  -451.8  921.65    89.9  864.63
   513.5  867.89    1272  914.64  1758.4  861.85  2164.9  927.45    2550  933.15
  2997.6  922.31  3236.2  868.83  3716.2  835.64  4421.6  780.73  4454.5  764.38
  5066.5  685.14    5366  776.72  5376.5   785.9    6256  813.85  8532.3  833.67
  9112.4  842.15  9465.2  843.25 10108.4  853.61 10553.9  943.19 10871.3  948.81
 11713.9  930.94   12198  955.95 12857.6  971.32 13880.2 1008.68 14418.6 1046.61
#Mann= 17 ,-1 , 0
 -1802.4     .05       0 -1745.4      .1       0    89.9      .1       0
   513.5     .16       0  3716.2     .16       0  4454.5    .035       0
  5376.5     .05       0    6256     .16       0  8532.3      .1       0
  9112.4      .1       0  9465.2     .05       0 10108.4     .16       0
 10871.3      .1       0 11713.9      .1       0   12198     .05       0
 12857.6      .1       0 13880.2     .16       0
Bank Sta=4421.6,5366
XS Rating Curve= 0 ,0
Exp/Cntr=0.3,0.1

Type RM Length L Ch R = 1 ,77429   ,2072,2072,2072
BEGIN DESCRIPTION:
PEDERNALES RIVER 304.0
END DESCRIPTION:
XS GIS Cut Line= 3
      2986449.34     10106784.64      2987027.73     10100021.03
      2995942.75     10095105.22
#Sta/Elev= 30
 -4554.1   951.6 -4533.8  951.11 -4133.3  941.37 -2805.4  882.61 -2074.2  912.16
 -1706.7  870.61 -1098.8  915.21  -423.2  850.69   749.8  826.26  2918.8  817.62
  3529.6  806.71    4656  805.21  4690.2  772.17  4699.7  772.14  4927.8  688.13
  5058.2  684.18  5427.5  774.41  5443.6  807.81  5685.6  814.71  6582.6  840.28
  6984.3  851.73  7902.2  883.54  8349.6     932  8674.8     932  9114.9  875.94
  9582.6  887.85 10036.7  931.76 10736.5  990.54 11911.7  996.72 12414.7 1034.18
#Mann= 19 ,-1 , 0
 -4554.1      .1       0 -4533.8     .16       0 -4133.3      .1       0
 -2805.4     .16       0 -1706.7      .1       0  -423.2     .05       0
   749.8     .05       0  2918.8     .05       0  3529.6     .05       0
  4690.2    .035       0  5443.6     .16       0  5685.6     .16       0
  6582.6     .05       0  6984.3     .05       0  7902.2      .1       0
  8349.6      .1       0  9582.6     .16       0 10036.7      .1       0
 10736.5      .1       0
Bank Sta=4699.7,5427.5
XS Rating Curve= 0 ,0
Exp/Cntr=0.3,0.1

Type RM Length L Ch R = 1 ,75357   ,2033,2033,2033
BEGIN DESCRIPTION:
PEDERNALES RIVER 305.0
END DESCRIPTION:
XS GIS Cut Line= 4
      2986975.23     10106374.53      2988169.17     10102483.05
      2993118.02      10098195.3      2996068.88       10095368.
#Sta/Elev= 30
 -2203.6  952.71 -1832.5  939.77  -895.5  884.96  -384.9  906.97   185.5  872.91
  1184.5  885.77  1707.6  923.48  2123.8   883.2  4358.5   809.2    4709  781.16
  4715.7  771.56    4949   682.8    5106  686.93  5425.2   773.5    5446   791.8
  5822.1  796.56  5906.6  759.51  5977.9  790.67  6212.9  798.46  7006.6  841.63
  7566.5  877.83  7820.4  929.44  8883.1 1002.31  9259.4 1002.47  9804.3   966.2
   10333  944.84   10877  991.31 12057.7 1035.83 12489.2 1050.88 12501.6 1051.49
#Mann= 19 ,-1 , 0
 -2203.6     .16       0 -1832.5     .05       0  -895.5      .1       0
  -384.9      .1       0   185.5      .1       0  1184.5      .1       0
  2123.8     .05       0  4358.5     .05       0  4715.7    .033       0
    5446     .16       0  6212.9      .1       0  7006.6     .05       0
  7566.5      .1       0  8883.1     .05       0  9259.4      .1       0
  9804.3      .1       0   10877      .1       0 12057.7      .1       0
 12489.2      .1       0
Bank Sta=4709,5425.2
XS Rating Curve= 0 ,0
Exp/Cntr=0.3,0.1

Type RM Length L Ch R = 1 ,73324   ,4157,4157,4157
BEGIN DESCRIPTION:
PEDERNALES RIVER 306.0
END DESCRIPTION:
XS GIS Cut Line= 4
      2987075.22     10106714.25      2989814.04     10102138.81
      2994150.46     10101046.62      2996299.19     10095760.73
#Sta/Elev= 30
 -2831.2  953.41 -2015.9  933.74 -1323.5  863.73 -1044.3  849.78  -291.8  832.16
     195  825.79   890.4  870.08  1280.6  865.84  2907.7  805.83  3924.6  791.58
  4507.4  783.41  4640.5  768.35  4650.8   757.2  4887.8  683.02  5114.9  688.53
  5367.6  758.89    5383  798.91  5951.7  849.47    6452  849.79  6981.4  856.72
  7219.7  899.36  7910.3  943.92  8433.6  921.24    8812  963.99    9250  947.05
  9982.2   932.6 10889.7  961.28 11625.8  964.02 12592.9 1023.88 12679.1 1028.56
#Mann= 19 ,-1 , 0
 -2831.2     .16       0 -2015.9     .05       0 -1323.5      .1       0
 -1044.3      .1       0  -291.8     .05       0     195     .05       0
   890.4      .1       0  1280.6     .05       0  2907.7      .1       0
  3924.6     .05       0  4507.4     .05       0  4640.5    .033       0
  5367.6     .16       0  5951.7     .05       0    6452      .1       0
    8812     .05       0    9250      .1       0 10889.7      .1       0
 12592.9     .16       0
Bank Sta=4650.8,5367.6
XS Rating Curve= 0 ,0
Exp/Cntr=0.3,0.1

Type RM Length L Ch R = 1 ,69167   ,2055,2055,2055
BEGIN DESCRIPTION:
PEDERNALES RIVER 307.0
END DESCRIPTION:
XS GIS Cut Line= 4
      2987254.86     10106924.86      2989489.64      10105207.7
       2994138.8     10104093.33      2996921.81     10098060.04
#Sta/Elev= 30
   770.1  942.45  1222.8  912.85  1467.6  924.15  2327.5  906.27  2731.5  917.59
  3587.6  839.07  4625.8  805.33    4667   768.3  4780.1  735.68  4869.3  684.19
  5084.2  683.01  5173.7  689.56  5438.2  764.26  6921.8  812.76    7630  831.07
  8511.5  852.49  8783.9  856.92  9249.9   864.5  9652.5  871.06 10189.2  890.09
 10748.5  923.89 11663.4  888.44 11865.7  870.71 12279.6  871.18 12560.2  880.79
 12874.4  902.08 13187.9  921.82 14141.4  967.84 14959.8 1001.42 15013.5 1003.62
#Mann= 19 ,-1 , 0
   770.1      .1       0  1467.6      .1       0  2731.5     .05       0
    4667    .033       0  5438.2     .05       0  6921.8     .05       0
    7630     .05       0  8511.5      .1       0  8783.9     .05       0
  9249.9     .05       0  9652.5     .16       0 10189.2     .16       0
 11663.4      .1       0 12279.6     .16       0 12560.2      .1       0
 12874.4     .16       0 13187.9      .1       0 14141.4     .16       0
 14959.8      .1       0
Bank Sta=4667,5438.2
XS Rating Curve= 0 ,0
Exp/Cntr=0.3,0.1

Type RM Length L Ch R = 1 ,67112   ,2010,2010,2010
BEGIN DESCRIPTION:
PEDERNALES RIVER 308.0
END DESCRIPTION:
XS GIS Cut Line= 4
      2987958.15     10111126.17      2993451.52     10104918.16
      2995396.66     10103457.86      2997075.45     10098270.27
#Sta/Elev= 30
 -1130.1  991.34  -759.3  970.84  -398.4  945.74   -95.3  946.13  1136.7  917.98
  1880.7  854.39  2080.8  834.52    3018  822.15  4285.5  811.06  4631.1  805.31
  4659.5     798  4667.1  760.39  4681.3  753.74  4914.4  683.93  5155.6  686.35
  5424.9  759.78  5467.6  784.24    5767  799.71  6728.4  819.52  8667.8  869.95
  9843.6  906.06 10540.9  925.76 11813.9  912.83 12055.6  904.34 12832.8  924.74
 13258.7  936.33 13618.5  945.02 14232.9  969.91 14874.2  988.17 15044.2   996.8
#Mann= 20 ,-1 , 0
 -1130.1     .16       0  -759.3      .1       0   -95.3     .16       0
  1136.7      .1       0  1880.7     .05       0    3018     .05       0
  4285.5     .16       0  4681.3    .033       0  5424.9     .05       0
    5767     .05       0  6728.4     .05       0  8667.8     .16       0
  9843.6      .1       0 10540.9     .16       0 11813.9      .1       0
 12832.8      .1       0 13258.7     .16       0 13618.5      .1       0
 14232.9     .16       0 14874.2      .1       0
Bank Sta=4667.1,5424.9
XS Rating Curve= 0 ,0
Exp/Cntr=0.3,0.1

Type RM Length L Ch R = 1 ,65102   ,2129,2129,2129
BEGIN DESCRIPTION:
PEDERNALES RIVER 309.0
END DESCRIPTION:
XS GIS Cut Line= 3
      2991618.75     10112030.85      2995496.94      10103771.6
      2997385.97     10098430.36
#Sta/Elev= 30
   116.7 1008.61   341.8  986.83   949.4   960.7    1546  895.39  1994.9  910.52
  2265.5  906.92  2398.1  882.49  2715.5  875.15  3295.2   828.6  4641.3  795.69
  4669.6  766.75  4676.2  759.22    4903  684.13  5142.4  689.17  5383.2  759.31
  5393.3  774.64  5593.6  793.14  5926.3  804.84  6495.2  815.22  7639.7  833.87
  8286.1  853.15  9446.4  900.95 10491.9  909.11 10909.9  919.17 11437.5  898.85
 12010.6  892.84 12289.1  913.34 13927.3  947.16 14603.1  959.12 14906.6  972.57
#Mann= 18 ,-1 , 0
   116.7     .05       0   341.8      .1       0    1546     .16       0
  1994.9      .1       0  2398.1      .1       0  4669.6    .033       0
  5393.3     .16       0  5593.6     .05       0  5926.3     .16       0
  6495.2     .05       0  7639.7     .05       0  8286.1     .16       0
  9446.4      .1       0 10491.9      .1       0 11437.5     .16       0
 12010.6      .1       0 13927.3      .1       0 14603.1     .16       0
Bank Sta=4676.2,5383.2
XS Rating Curve= 0 ,0
Exp/Cntr=0.3,0.1

Type RM Length L Ch R = 1 ,62973   ,1505,1505,1505
BEGIN DESCRIPTION:
PEDERNALES RIVER 310.0
END DESCRIPTION:
XS GIS Cut Line= 4
      2991746.05     10112266.76      2995425.74     10109525.87
      2997276.26     10100981.13      2997759.19     10097731.86
#Sta/Elev= 30
  -732.7 1015.06   489.9  914.21    1041  905.72  1593.4  903.54  1849.7  871.75
  2644.4   827.3  2936.3   847.4  3319.6  842.87  3886.5  819.02  4649.4   785.6
  4686.6  746.45    4707  733.63  4911.4  683.83    5147  684.98  5351.6  749.04
  5361.9  747.79  5392.6  785.39  5970.8  803.28    6590  783.82  6953.9  801.25
    7863  807.16  8572.2  826.78  9497.5  824.57 10146.6  832.11 11663.4  850.09
 12061.6   859.6 13038.2   887.6 14831.5  940.72 15250.1  961.09 15883.4  977.66
#Mann= 18 ,-1 , 0
  -732.7      .1       0   489.9      .1       0    1041      .1       0
  1849.7     .16       0  3319.6     .05       0  3886.5      .1       0
    4707    .033       0  5361.9     .05       0  6953.9     .05       0
    7863      .1       0  8572.2     .16       0  9497.5     .05       0
 10146.6     .05       0 11663.4      .1       0 12061.6      .1       0
 13038.2      .1       0 14831.5      .1       0 15250.1      .1       0
Bank Sta=4686.6,5351.6
XS Rating Curve= 0 ,0
Exp/Cntr=0.3,0.1

Type RM Length L Ch R = 1 ,61468   ,3257,3257,3257
BEGIN DESCRIPTION:
PEDERNALES RIVER 311.0
END DESCRIPTION:
XS GIS Cut Line= 4
      2991844.61       10112485.      2996301.56     10110066.22
      2998996.23     10106258.47      3000863.52     10099163.76
#Sta/Elev= 30
 -1352.4  990.27    87.6  867.56   892.1  854.72  1298.9  837.11  1798.4  815.84
  2501.1  795.56  2898.6   786.2  3482.3  814.74  4088.5  795.37  4529.8  763.31
  4535.9  761.14  4664.9  718.64  4901.4  684.33  5180.8  684.84  5311.3  712.82
  5468.6  683.48    5763  763.35  5769.1  768.99  5804.8  787.27  7181.2     819
  8213.7  843.85  8628.6  841.74  9056.5  828.89  9645.3  850.19 10148.1  898.83
 11120.3  956.22   12461  990.74 13856.6  987.59   15135  994.06 15719.7  1019.1
#Mann= 19 ,-1 , 0
 -1352.4      .1       0    87.6     .16       0   892.1      .1       0
  1298.9     .05       0  1798.4     .16       0  2501.1     .16       0
  4088.5     .16       0  4529.8    .033       0    5763     .16       0
  7181.2     .16       0  8213.7      .1       0  8628.6     .05       0
  9056.5     .16       0  9645.3      .1       0 10148.1      .1       0
 11120.3     .16       0   12461      .1       0 13856.6      .1       0
   15135     .16       0
Bank Sta=4535.9,5769.1
XS Rating Curve= 0 ,0
Exp/Cntr=0.3,0.1

Type RM Length L Ch R = 1 ,58211   ,1653,1653,1653
BEGIN DESCRIPTION:
PEDERNALES RIVER 312.0
END DESCRIPTION:
XS GIS Cut Line= 4
      2991579.46     10112872.32       2995653.8     10111555.57
      2999900.91     10112063.86      3000824.29      10104089.3
#Sta/Elev= 30
   -1335  981.14 -1198.6  968.77  -771.1  961.87  -324.5  946.01   556.7  871.59
  1047.1  839.99  3636.4  791.43  3726.4  771.93  4089.6  791.69    4318  754.86
  4323.1  754.84  4804.4  683.07  5217.6  686.52  5459.3  758.14  5479.4  784.06
  6144.2  809.84  7133.1  848.19  8519.1  812.49  9509.9  839.33 10100.9  855.35
 10494.9  879.98 11334.7  916.31 11692.1  884.86 12177.3  884.52 12813.6  965.67
 13272.5  963.16 13780.1  944.88   14238  959.48 14944.9  965.66 15252.1  968.35
#Mann= 18 ,-1 , 0
   -1335      .1       0 -1198.6     .16       0  -771.1     .16       0
  -324.5      .1       0   556.7     .05       0  1047.1     .16       0
  4323.1    .033       0  6144.2     .05       0  7133.1     .05       0
  8519.1      .1       0  9509.9     .16       0 10100.9     .16       0
 10494.9      .1       0 11692.1      .1       0 13272.5     .16       0
 13780.1     .16       0   14238     .05       0 14944.9     .16       0
Bank Sta=4318,5459.3
XS Rating Curve= 0 ,0
Exp/Cntr=0.3,0.1

Type RM Length L Ch R = 1 ,56558   ,1997,1997,1997
BEGIN DESCRIPTION:
PEDERNALES RIVER 313.0
END DESCRIPTION:
XS GIS Cut Line= 3
      2991422.98     10113239.31      2999928.19     10113366.26
      3000982.13     10107108.25
#Sta/Elev= 30
  -701.9  979.02  -643.8  977.79   263.6  917.78  1318.1  853.06  1963.9  868.66
  2156.9  892.13  2303.9  891.36  2600.4  839.76  3192.3  808.24  3783.5  800.59
  4423.8  796.53  4624.4  770.41  4634.2  743.04  4824.2  684.44    4974  683.59
  5194.2  686.67  5444.3  756.81  5464.3  766.52  5959.5  794.33  7433.8  819.22
  7703.2  816.72  8749.2  878.23  9632.2  866.14  9926.9  836.92 10152.5  827.92
 11015.9  842.09 11538.1  854.95 12185.8  879.03 13039.5  930.79 14150.4  948.87
#Mann= 19 ,-1 , 0
  -701.9     .16       0  -643.8      .1       0   263.6     .16       0
  1318.1     .16       0  2156.9     .05       0  2600.4     .05       0
  3192.3     .16       0  3783.5      .1       0  4423.8     .16       0
  4634.2    .033       0  5444.3     .16       0  7433.8      .1       0
  7703.2     .16       0  8749.2     .05       0  9926.9     .05       0
 10152.5      .1       0 11015.9     .16       0 11538.1      .1       0
 12185.8      .1       0
Bank Sta=4624.4,5464.3
XS Rating Curve= 0 ,0
Exp/Cntr=0.3,0.1

Type RM Length L Ch R = 1 ,54561   ,1876,1876,1876
BEGIN DESCRIPTION:
PEDERNALES RIVER 314.0
END DESCRIPTION:
XS GIS Cut Line= 5
      2992458.01     10115530.71      2996059.51     10115596.97
      2999106.31     10114896.85      3000698.62     10112486.06
      3001010.85     10108301.59
#Sta/Elev= 30
    79.2  984.54   140.4   983.9  1029.8  874.04  1472.1  841.79  2052.7  823.96
  2421.2  815.92  3185.8  798.76  3734.5  780.62  4049.6  760.47  4059.9   756.2
  4316.4   684.9  4700.8   706.4  4849.7   683.2  5198.8  684.67    5404  754.21
  5417.2  768.41  5434.8  746.39    5460  760.97  5465.6  792.39  5545.7  798.74
  6389.9  807.97  6696.7  802.69    7414  803.79  8133.1   797.2  9239.9  839.99
  9495.3  844.27 10301.9  841.49 11677.9   845.9 12456.1   883.2 13892.8  921.06
#Mann= 18 ,-1 , 0
    79.2     .16       0   140.4      .1       0  1472.1     .05       0
  2052.7      .1       0  2421.2     .16       0  3185.8     .05       0
  3734.5     .16       0  4059.9    .033       0  5434.8     .16       0
  6389.9     .16       0  6696.7     .05       0    7414     .16       0
  8133.1     .16       0  9239.9      .1       0  9495.3     .05       0
 10301.9     .16       0 11677.9     .16       0 12456.1      .1       0
Bank Sta=4049.6,5404
XS Rating Curve= 0 ,0
Exp/Cntr=0.3,0.1

Type RM Length L Ch R = 1 ,52685   ,2230,2230,2230
BEGIN DESCRIPTION:
PEDERNALES RIVER 315.0
END DESCRIPTION:
XS GIS Cut Line= 4
      2996974.94     10118913.86      2998692.75     10115347.45
      3000833.65       10113499.      3001311.29     10108574.43
#Sta/Elev= 30
  2949.3  883.69  3334.8   837.1  3793.8  814.17  4143.4  796.75  4241.1  776.82
  4284.7  796.63    4426  796.02  4465.7  761.41    4570  738.27  4592.2  726.11
  4765.3  685.52  5115.5  682.93  5380.2   687.3  5505.8  736.52  5709.4  760.73
    6181  763.81    6631  796.52  6914.9  802.58  7437.5  799.53  8646.3  786.16
  9375.3   799.2  9874.2  812.73 11054.8  840.82   11709  821.79 11986.2  820.18
 12432.1  825.76 13120.8  866.01 13708.2  894.34 14463.7  939.59   14684  933.47
#Mann= 18 ,-1 , 0
  2949.3      .1       0  3334.8     .05       0  3793.8     .05       0
  4241.1     .16       0  4592.2    .033       0  5505.8     .16       0
    6181      .1       0  6914.9     .16       0  7437.5     .05       0
  8646.3     .16       0  9375.3     .05       0  9874.2     .16       0
 11054.8     .16       0   11709     .05       0 11986.2     .16       0
 12432.1     .05       0 13120.8     .16       0 13708.2      .1       0
Bank Sta=4570,5505.8
XS Rating Curve= 0 ,0
Exp/Cntr=0.3,0.1

Type RM Length L Ch R = 1 ,50455   ,2148,2148,2148
BEGIN DESCRIPTION:
PEDERNALES RIVER 316.0
END DESCRIPTION:
XS GIS Cut Line= 5
      2998101.07     10119101.42      3000297.76     10117520.05
      2999290.49     10115094.44      3001266.33     10113256.96
      3001413.72     10108714.58
#Sta/Elev= 30
   759.6  888.26   910.7  884.19  1092.3  851.51  1415.1  832.41  2699.2  819.09
    2980  811.25  3407.3  798.25  4061.8  796.29  4450.6  778.52  4548.5  772.87
  4555.9  770.45  4642.6  720.37  4779.3  683.71    5247  684.57  5536.6   756.9
  5552.1  769.18  5907.4  791.63  6247.5  776.67    6502  790.31  7181.7   782.8
  7237.7  762.99  7393.7  783.84  8497.4  810.09  8877.7  804.46   10185  818.79
 11084.5  817.67   11714  849.26 12008.7  864.88 12674.2  899.01 13335.7   940.9
#Mann= 18 ,-1 , 0
   759.6      .1       0   910.7     .05       0  2699.2     .16       0
    2980     .05       0  3407.3     .16       0  4061.8     .05       0
  4450.6     .16       0  4548.5    .033       0  5536.6     .16       0
  5907.4     .05       0    6502     .05       0  7237.7     .16       0
  8877.7     .16       0   10185     .05       0 11084.5     .16       0
   11714      .1       0 12008.7     .16       0 12674.2      .1       0
Bank Sta=4555.9,5552.1
XS Rating Curve= 0 ,0
Exp/Cntr=0.3,0.1

Type RM Length L Ch R = 1 ,48307   ,1574,1574,1574
BEGIN DESCRIPTION:
PEDERNALES RIVER 317.0
END DESCRIPTION:
XS GIS Cut Line= 5
      3004042.89     10117053.53      3002069.05     10116629.79
      3001114.03     10113840.24      3001701.47     10112666.98
      3001505.83      10108846.9
#Sta/Elev= 30
  1133.6  890.04  1236.4   887.3  1400.6  883.22  1584.1  880.36  1875.4  860.74
    1983  844.54  2536.8  813.93  3301.2  795.77  4183.6  781.53  4402.7  765.84
  4416.6  761.87  4659.7  696.54  4754.6  683.06  5174.4  686.25  5251.6  719.26
  5283.3  720.85  5315.1  748.72  5325.6  782.76  5528.1  794.42  5802.8  795.76
  6175.5  804.71  6703.4  800.25  6913.3  799.82  7910.8  806.98    8357  805.85
    8768   803.8  9975.2  853.57   10818   900.9 11068.8  913.08 11238.1  925.82
#Mann= 18 ,-1 , 0
  1133.6     .16       0  1236.4      .1       0  1400.6     .05       0
    1983     .05       0  2536.8     .05       0  3301.2     .16       0
  4416.6    .033       0  5315.1     .16       0  5528.1     .05       0
  5802.8     .05       0  6175.5     .16       0  6703.4     .05       0
  6913.3     .16       0  7910.8     .05       0    8357     .16       0
  9975.2     .16       0   10818     .16       0 11068.8      .1       0
Bank Sta=4402.7,5325.6
XS Rating Curve= 0 ,0
Exp/Cntr=0.3,0.1

Type RM Length L Ch R = 1 ,46733   ,1492,1492,1492
BEGIN DESCRIPTION:
PEDERNALES RIVER 318.0
END DESCRIPTION:
XS GIS Cut Line= 3
       3004257.1     10116930.28      3001893.71     10112213.64
      3001675.87     10108778.27
#Sta/Elev= 30
  1964.5  891.13  2124.7  886.19  2304.6  878.96  2395.3  864.05  2564.6  854.28
  2617.5  839.86  2790.2  825.75    2957  817.32  3557.9  796.04  4080.4  780.21
  4315.8  780.98  4388.4  771.97  4405.2  766.97  4500.1  716.92  4790.4  683.59
  5226.4  684.97  5260.3  703.43  5410.8  759.34  5416.9  761.66  5854.1  789.19
  6869.9  794.14  7194.8  800.53  7634.9   801.9  8189.5  801.43  8934.3  828.51
  9203.4  840.61  9499.8  852.11 10466.3  907.84 10661.7  914.73 10682.4  915.38
#Mann= 18 ,-1 , 0
  1964.5     .16       0  2124.7     .16       0  2395.3     .05       0
  2790.2      .1       0    2957     .05       0  3557.9     .16       0
  4080.4     .16       0  4388.4    .033       0  5410.8     .16       0
  5854.1     .05       0  6869.9     .05       0  7194.8     .05       0
  7634.9     .16       0  8934.3     .05       0  9203.4     .16       0
  9499.8     .16       0 10466.3      .1       0 10661.7     .05       0
Bank Sta=4405.2,5416.9
XS Rating Curve= 0 ,0
Exp/Cntr=0.3,0.1

Type RM Length L Ch R = 1 ,45241   ,2218,2218,2218
BEGIN DESCRIPTION:
PEDERNALES RIVER 319.0
END DESCRIPTION:
XS GIS Cut Line= 4
      3004544.98     10116816.71      3004493.23     10113986.26
      3002637.96     10110994.58      3001764.34     10108640.01
#Sta/Elev= 30
  1378.4  886.86  1629.9  880.03  2071.5  836.58  2358.5  821.65  3007.3  807.62
  3501.7  793.16  3696.6  797.55  4475.8  781.48  4664.8   767.8  4707.3  723.16
  4783.8  687.55  4897.2  685.01  5228.8  683.69  5231.6  683.19  5234.8  683.69
  5426.7  715.69  5536.6   773.5  5728.7  785.91    5865  790.35  6298.9   799.5
  6887.5  799.78  7089.4  792.06  7243.5  785.32  7629.5  796.48  7929.8  802.22
  8203.4   810.2  8811.7  831.57  9117.8  843.92 10090.2  907.51   10241  908.87
#Mann= 20 ,-1 , 0
  1378.4     .05       0  1629.9     .16       0  2358.5     .05       0
  3007.3     .16       0  3696.6     .16       0  4783.8     .07       0
  4897.2     .05       0  5228.8    .033       0  5234.8     .16       0
  5728.7     .16       0    5865     .05       0  6298.9      .1       0
  6887.5     .05       0  7089.4     .16       0  7629.5     .16       0
  7929.8     .05       0  8203.4     .16       0  8811.7     .05       0
  9117.8     .16       0 10090.2      .1       0
Bank Sta=5228.8,5234.8
XS Rating Curve= 0 ,0
Exp/Cntr=0.3,0.1

Type RM Length L Ch R = 1 ,43023   ,1877,1877,1877
BEGIN DESCRIPTION:
PEDERNALES RIVER 329.0
END DESCRIPTION:
XS GIS Cut Line= 3
      3006222.49     10116811.77      3005994.28      10113371.5
      3006368.23     10106730.35
#Sta/Elev= 30
   742.9  872.89    1216  859.79  1413.6  851.26  1757.3  825.27  2015.9  812.49
  2696.2  785.49  2994.6  788.85  3389.8  793.61  4081.5  777.99  4376.9  761.33
  4776.4  684.16  4779.2  683.66  4782.4  684.16  4879.3   688.8  5244.3  684.68
  5350.3  722.21  5370.4  773.02  5457.6   780.6  6047.1  795.69  6323.6   802.8
  7913.7  830.05  8601.5  814.59    8980  797.04  9583.9  828.02  9817.4     833
  9897.5  855.93 10084.2  861.89 10288.1  884.41 10762.9  899.89 10842.4  900.95
#Mann= 20 ,-1 , 0
   742.9      .1       0    1216     .16       0  1413.6     .05       0
  1757.3     .16       0  2015.9     .05       0  2994.6     .16       0
  3389.8     .05       0  4081.5     .05       0  4376.9      .1       0
  4776.4    .033       0  4782.4      .1       0  4879.3     .05       0
  5457.6     .08       0  6047.1     .16       0  6323.6     .16       0
  7913.7     .16       0  8601.5     .16       0  9583.9     .05       0
 10084.2     .16       0 10762.9      .1       0
Bank Sta=4776.4,4782.4
XS Rating Curve= 0 ,0
Exp/Cntr=0.3,0.1

Type RM Length L Ch R = 1 ,41146   ,1749,1749,1749
BEGIN DESCRIPTION:
PEDERNALES RIVER 330.0
END DESCRIPTION:
XS GIS Cut Line= 3
      3006366.74     10116938.56      3007711.54     10114330.26
      3008664.16     10106383.83
#Sta/Elev= 30
   657.2  869.99   702.4  868.79  1018.7  860.76  2176.3   825.1  2556.7  813.54
  3135.7  792.01  3681.5  785.39  4174.2  781.24  4666.8  750.34  4695.6  714.38
  4863.9  685.55  5166.5  684.06  5169.3  683.56  5172.5  684.06  5278.5  691.67
  5401.2  716.04  5421.3  771.05  5431.4   773.9  5849.2  782.53  6539.3  816.35
  6986.2  866.68  7224.9  888.32  8016.8  889.89  8232.5  906.67    8608  887.49
  9464.1   839.3   10024  865.95 10677.2  934.59 11071.3  949.74 11595.1  958.47
#Mann= 20 ,-1 , 0
   657.2      .1       0   702.4     .05       0  1018.7     .16       0
  2176.3     .16       0  2556.7      .1       0  3135.7     .16       0
  3681.5     .05       0  4174.2     .16       0  4666.8     .16       0
  4863.9     .05       0  5166.5    .033       0  5172.5     .05       0
  5278.5     .16       0  5849.2     .16       0  6986.2      .1       0
  8016.8      .1       0    8608     .05       0  9464.1     .16       0
 10677.2     .16       0 11071.3     .16       0
Bank Sta=5166.5,5172.5
XS Rating Curve= 0 ,0
Exp/Cntr=0.3,0.1

Type RM Length L Ch R = 1 ,39397   ,2214,2214,2214
BEGIN DESCRIPTION:
PEDERNALES RIVER 321.0
END DESCRIPTION:
XS GIS Cut Line= 4
      3006154.57     10117248.42      3008311.73     10114650.19
      3010521.31     10112865.11      3012001.36     10111112.63
#Sta/Elev= 30
   357.4  870.19   736.5  866.94  1088.8   854.3  1414.3   841.9  1747.4  829.21
  1994.4   819.8  2169.1  813.14  2502.8  805.77  2683.4  802.32  3042.2  792.33
  3530.5  776.78  3869.5  766.33  4611.4  744.45  4782.4  683.97  4864.2  683.71
    4867  683.21  4870.2  683.71  4891.7  683.76  5277.5  688.88  5337.2  712.73
  5358.1   767.1    5803  788.63  6623.7  862.26  7013.7  871.16  7311.5  957.88
  7504.4  983.08  7952.9  949.97  8150.1  973.32  8745.5 1020.71  8868.8 1054.57
#Mann= 20 ,-1 , 0
   357.4      .1       0   736.5     .05       0  1088.8     .16       0
  1414.3     .05       0  1747.4     .16       0  1994.4     .05       0
  2169.1     .16       0  2502.8     .16       0  2683.4      .1       0
  3042.2     .16       0  3530.5      .1       0  3869.5     .16       0
  4864.2    .033       0  4870.2      .1       0  4891.7     .05       0
  5277.5     .16       0    5803     .16       0  7504.4      .1       0
  7952.9     .16       0  8150.1      .1       0
Bank Sta=4864.2,4870.2
XS Rating Curve= 0 ,0
Exp/Cntr=0.3,0.1

Type RM Length L Ch R = 1 ,37183   ,2959,2959,2959
BEGIN DESCRIPTION:
PEDERNALES RIVER 322.0
END DESCRIPTION:
XS GIS Cut Line= 3
      3006212.64      10117603.3       3012622.7     10114766.13
      3013964.35     10113909.28
#Sta/Elev= 30
   310.7  872.09   614.8  853.37    1604  840.86  2050.4  814.92  2715.8  788.74
    2845  783.94    3473  775.57    3693  774.36    4522   736.3  4672.7  747.04
  4791.6  684.46  4794.4  683.96  4797.6  684.46  4902.8  684.61  5307.3  701.37
  5357.6  716.94  5402.2  765.93  5545.9  797.25  5672.7  820.59  5879.5  872.72
  6112.6  888.53  6332.6  910.65  6487.1  923.63  6894.5  957.12  7176.3  925.42
  7790.2  832.28  8188.3   947.9  8561.9   993.9  8897.4 1038.09  8912.5 1038.61
#Mann= 20 ,-1 , 0
   310.7      .1       0   614.8     .16       0    1604     .05       0
  2050.4     .05       0  2715.8      .1       0    2845     .16       0
    3473     .05       0    3693     .16       0  4791.6    .033       0
  4797.6     .16       0  4902.8     .05       0  5307.3     .16       0
  5545.9     .08       0  5672.7     .16       0  6112.6      .1       0
  6332.6      .1       0  6487.1      .1       0  7176.3     .16       0
  8561.9     .05       0  8897.4     .16       0
Bank Sta=4791.6,4797.6
XS Rating Curve= 0 ,0
Exp/Cntr=0.3,0.1

Type RM Length L Ch R = 1 ,34224   ,2044,2044,2044
BEGIN DESCRIPTION:
PEDERNALES RIVER 323.0
END DESCRIPTION:
XS GIS Cut Line= 3
      3005959.42     10117870.97      3008751.57     10117822.24
      3013641.82     10119945.32
#Sta/Elev= 30
   637.9  874.37  1079.5  857.57  1286.2  844.49  1502.7  826.16  1833.3  812.84
  2254.2  812.86  2571.5  802.82  3424.6  787.85    3846  773.47    4163  764.14
  4495.5  746.19  4696.7  683.56  4699.5  683.06  4702.7  683.56  5247.7  683.95
  5282.9   713.5  5313.1  709.78  5329.8  755.65  5348.9  758.71    5589  762.71
  5761.2  745.49    5884  769.46  6032.8  778.14    7227  821.54  7308.1  815.31
  7853.8  860.77  8017.4  870.39  8162.9  884.38  8602.7  935.47  8761.7  940.39
#Mann= 20 ,-1 , 0
   637.9     .05       0  1079.5     .16       0  1286.2      .1       0
  1502.7      .1       0  1833.3     .16       0  2254.2      .1       0
  2571.5     .16       0  3424.6     .16       0    3846      .1       0
    4163     .05       0  4696.7    .033       0  4702.7     .05       0
  5348.9     .05       0    5589     .16       0  6032.8     .05       0
    7227     .16       0  7853.8     .05       0  8017.4     .08       0
  8162.9     .05       0  8602.7     .08       0
Bank Sta=4696.7,4702.7
XS Rating Curve= 0 ,0
Exp/Cntr=0.3,0.1

Type RM Length L Ch R = 1 ,32180   ,2465,2465,2465
BEGIN DESCRIPTION:
PEDERNALES RIVER 324.0
END DESCRIPTION:
XS GIS Cut Line= 3
      3005832.31     10118036.04      3007128.59     10119343.76
      3013782.04     10122071.97
#Sta/Elev= 30
  1106.1  871.28  1336.3  858.54  1957.4   827.8  2544.3  832.48  2745.5  838.34
  3224.5  805.49    3836  785.91  4491.5  760.93  4636.1  754.81  4648.5  753.24
    4655  725.55  4665.8     709    4760  683.73  4762.8  683.23    4766  683.73
  4806.1  683.75  5247.8  684.15  5325.1  694.52  5422.3  741.58  5644.9  763.97
  5791.2  765.36  6064.3  769.03  6406.4  781.27  6903.2  804.56  7279.6  834.92
  7797.8  850.47  7951.7  852.67  8787.4  826.48 10122.7   912.2 10138.5  912.71
#Mann= 20 ,-1 , 0
  1106.1     .05       0  1336.3     .16       0  2544.3      .1       0
  2745.5      .1       0  3224.5      .1       0    3836      .1       0
  4491.5      .1       0  4636.1     .16       0    4760    .033       0
    4766     .16       0  4806.1     .05       0  5247.8     .16       0
  5644.9     .08       0  5791.2     .16       0  6064.3     .05       0
  6406.4     .05       0  6903.2     .16       0  7797.8     .05       0
  7951.7     .16       0 10122.7      .1       0
Bank Sta=4760,4766
XS Rating Curve= 0 ,0
Exp/Cntr=0.3,0.1

Type RM Length L Ch R = 1 ,29715   ,3060,3060,3060
BEGIN DESCRIPTION:
PEDERNALES RIVER 325.0
END DESCRIPTION:
XS GIS Cut Line= 4
      3005016.01     10118345.37      3006055.87     10121292.22
      3012075.05     10124491.72      3013727.52     10124234.43
#Sta/Elev= 30
  -579.2  861.32   348.7  850.98     614   848.1  1276.7  840.91  1944.5   826.7
  2182.8  815.11  2738.3  792.68  2847.6  791.12  4450.7  755.91  4575.8  743.81
  4604.5   715.7  4708.8  684.72  4859.6  683.89  4862.4  683.39  4865.6  683.89
  5252.6  684.26  5367.4  693.02  5499.3  746.69  5565.2  756.73  6598.7  775.16
  6937.2  778.59  7513.6  783.22  8094.9  801.76  8584.1  809.13  9297.4  834.95
  9564.6  832.14  9704.7  829.15   10107   834.2 10750.7  867.94 11034.8  901.52
#Mann= 20 ,-1 , 0
  -579.2     .05       0   348.7      .1       0     614     .05       0
  1276.7      .1       0  1944.5     .05       0  2182.8     .05       0
  2738.3      .1       0  2847.6     .05       0  4859.6    .033       0
  4865.6     .05       0  5252.6     .16       0  6598.7     .05       0
  6937.2     .05       0  7513.6      .1       0  8094.9     .16       0
  9297.4     .05       0  9564.6     .05       0  9704.7     .16       0
   10107     .16       0 10750.7      .1       0
Bank Sta=4859.6,4865.6
XS Rating Curve= 0 ,0
Exp/Cntr=0.3,0.1

Type RM Length L Ch R = 1 ,26655   ,1334,1334,1334
BEGIN DESCRIPTION:
PEDERNALES RIVER 326.0
END DESCRIPTION:
XS GIS Cut Line= 3
      3004755.43     10118359.49      3004960.33      10122841.1
      3008072.65     10126629.11
#Sta/Elev= 30
 -1237.5  858.22  -977.6  849.95  -705.3  843.89  1117.6   799.9  1418.4  796.53
  1733.8  793.59  2198.3  791.42  2375.7  790.46  2888.6  787.67  3869.6   766.1
    4048  760.51  4357.6  747.83  4464.5  705.19  4548.3  700.92  4620.9  684.38
  5320.4  683.68  5323.1  683.18  5326.4  683.68  5423.8   722.7  5452.4  711.37
    5459  737.57  5473.3  753.34  5717.8  762.43  6084.6  748.83  6457.2  764.93
  6625.8  761.89  7248.6  766.67  7712.8  785.98  8039.4   802.3  8151.4  808.23
#Mann= 20 ,-1 , 0
 -1237.5     .16       0  -977.6     .16       0  -705.3     .05       0
  1117.6      .1       0  1418.4      .1       0  1733.8     .05       0
  2198.3      .1       0  2375.7     .05       0  2888.6     .16       0
  3869.6     .05       0    4048     .16       0  4548.3     .05       0
  5320.4    .033       0  5326.4     .16       0  5717.8     .16       0
  6457.2      .1       0  6625.8     .16       0  7248.6     .05       0
  7712.8      .1       0  8039.4     .05       0
Bank Sta=5320.4,5326.4
XS Rating Curve= 0 ,0
Exp/Cntr=0.3,0.1

Type RM Length L Ch R = 1 ,25321   ,2310,2310,2310
BEGIN DESCRIPTION:
PEDERNALES RIVER 327.0
END DESCRIPTION:
XS GIS Cut Line= 5
      3000920.34     10118928.29       3002964.3     10122104.59
      3004273.48     10123631.17       3006337.3     10127302.45
      3007744.82     10127085.75
#Sta/Elev= 30
 -1849.9  868.74 -1664.5  869.19 -1198.1  835.77     -49  802.59   513.2  797.49
   891.6  793.22  1197.8  785.45  2645.7  751.93  2681.1  723.13  2773.3  693.15
  2908.3  684.23  3099.3  753.99  3189.8  757.08  4178.8  779.14  4552.7  767.04
  4590.3  717.03  4758.8  684.27  5359.4  683.98  5362.1  683.48  5365.4  683.98
  5573.4  704.25  5794.6  701.92  6250.7  761.68  6503.6  778.92  6862.2  786.04
  7129.1  790.77  7463.7  795.12  8944.1  782.01  9490.4  796.52    9574  799.39
#Mann= 20 ,-1 , 0
 -1849.9     .08       0 -1664.5     .05       0 -1198.1     .05       0
     -49     .05       0   513.2     .16       0   891.6      .1       0
  1197.8     .05       0  2645.7     .16       0  3189.8     .05       0
  4178.8     .16       0  4758.8     .05       0  5359.4    .033       0
  5365.4     .16       0  6250.7     .08       0  6503.6     .05       0
  6862.2     .05       0  7129.1     .08       0  7463.7     .05       0
  8944.1      .1       0  9490.4      .1       0
Bank Sta=5359.4,5365.4
XS Rating Curve= 0 ,0
Exp/Cntr=0.3,0.1
