--- CALOHAN CREEK.prj (project) ---

Proj Title=CALOHAN CREEK Base Level Engineering
Current Plan=p01
Default Exp/Contr=0.3,0.1
English Units
Geom File=g01
Flow File=f01
Plan File=p01
Y Axis Title=Elevation
X Axis Title(PF)=Main Channel Distance
X Axis Title(XS)=Station
BEGIN DESCRIPTION:
CALOHAN CREEK
END DESCRIPTION:
DSS Export Rating Curves= 0
DSS Export Rating Curve Sorted= 0
DSS Export Volume Flow Curves= 0
DXF OffsetX= 0
DXF OffsetY= 0
DXF ScaleX= 1
DXF ScaleY= 10

--- CALOHAN CREEK.p01 (plan) ---

Plan Title=Multiple Run
Short Identifier=Multiple
Geom File=g01
Flow File=f01
Subcritical Flow
K Sum by GR= 0
Std Step Tol= 0.01
Critical Tol= 0.01
Num of Std Step Trials= 20
Max Error Tol= 0.3
Flow Tol Ratio= 0.001
Split Flow NTrial= 30
Split Flow Tol= 0.02
Split Flow Ratio= 0.02
Log Output Level= 0
Friction Slope Method= 1
Unsteady Friction Slope Method= 2
Unsteady Bridges Friction Slope Method= 1
Parabolic Critical Depth
Global Vel Dist=  1 , 1 , 1
Global Log Level= 0
CheckData=True
Encroach Param= -1, 0, 0, 0
BEGIN DESCRIPTION:
Multiple Run
END DESCRIPTION:

--- CALOHAN CREEK.f01 (steady flow) ---

Flow Title=Multiple
Program Version=4.10
Number of Profiles= 7
Profile Names=10-year,25-year,50-year,1pct_min,100-year,1pct_plu,500-year
River Rch & RM=CALOHAN CREEK,Reach-1         ,29737
    1085    1601    2058    1938    2622    3545    4268
River Rch & RM=CALOHAN CREEK,Reach-1         ,27278
    1188    1755    2257    2127    2876    3889    4683
River Rch & RM=CALOHAN CREEK,Reach-1         ,24305
    1356    2015    2601    2457    3323    4493    5442
River Rch & RM=CALOHAN CREEK,Reach-1         ,21829
    1472    2192    2834    2680    3625    4902    5951
River Rch & RM=CALOHAN CREEK,Reach-1         ,19644
    2286    3471    4547    4349    5882    7954    9882
River Rch & RM=CALOHAN CREEK,Reach-1         ,18521
    2286    3471    4547    4349    5882    7954    9882
River Rch & RM=CALOHAN CREEK,Reach-1         ,12852
    2682    4095    5383    5164    6983    9444   11803
River Rch & RM=CALOHAN CREEK,Reach-1         ,8769
    2916    4464    5878    5645    7635   10325   12936
River Rch & RM=CALOHAN CREEK,Reach-1         ,6699
    3029    4632    6094    5846    7906   10691   13363
Boundary for River Rch & Prof#=CALOHAN CREEK,Reach-1         , 1
Up Type= 0
Dn Type= 3
Dn Slope=0.005
Boundary for River Rch & Prof#=CALOHAN CREEK,Reach-1         , 2
Up Type= 0
Dn Type= 3
Dn Slope=0.005
Boundary for River Rch & Prof#=CALOHAN CREEK,Reach-1         , 3
Up Type= 0
Dn Type= 3
Dn Slope=0.005
Boundary for River Rch & Prof#=CALOHAN CREEK,Reach-1         , 4
Up Type= 0
Dn Type= 3
Dn Slope=0.005
Boundary for River Rch & Prof#=CALOHAN CREEK,Reach-1         , 5
Up Type= 0
Dn Type= 3
Dn Slope=0.005
Boundary for River Rch & Prof#=CALOHAN CREEK,Reach-1         , 6
Up Type= 0
Dn Type= 3
Dn Slope=0.005
Boundary for River Rch & Prof#=CALOHAN CREEK,Reach-1         , 7
Up Type= 0
Dn Type= 3
Dn Slope=0.005
DSS Import GetInterval= 0
DSS Import GetPeak= 0
DSS Import FillOption= 0

--- CALOHAN CREEK.g01 (geometry) ---

Geom Title=Existing Conditions
Program Version=4.10

River Reach=CALOHAN CREEK   ,Reach-1
Reach XY= 30
      2965815.87     10043814.15      2965224.89     10044756.14
      2964360.76     10044784.68      2964156.05     10046432.67
      2963814.99      10047100.1      2963936.23     10047408.45
      2962830.93     10048314.75       2962549.5     10049064.35
      2962670.99     10049511.32      2961808.24     10049677.45
      2962043.56     10050486.31      2961091.43     10050944.97
       2960849.8     10052104.02       2961269.1     10053035.52
      2960975.76     10053433.71      2961131.65     10054426.99
      2960848.59     10055454.59      2961088.47     10056293.73
      2960788.22     10057536.91      2961275.67     10057980.18
      2960546.64     10058586.42      2960248.48     10059217.33
      2960096.43     10060987.94      2959591.61     10061431.18
      2959575.59     10062262.54      2958929.21     10064078.99
      2959377.63     10064654.16      2959283.12     10066326.52
      2960142.37     10066865.89      2960138.47     10067143.73

Type RM Length L Ch R = 1 ,29737   ,540,540,540
BEGIN DESCRIPTION:
CALOHAN CREEK 65.0
END DESCRIPTION:
XS GIS Cut Line= 4
      2965591.65     10043647.93      2965674.96     10043807.61
      2965942.33     10044085.39      2966573.88     10044238.07
#Sta/Elev= 30
  4693.9 1284.69  4753.4 1279.08  4909.2 1269.09  4930.3 1260.77  4944.5 1257.12
  4979.7 1253.82  4998.1 1251.09  5000.8 1250.59  5004.1 1251.09  5022.1  1253.8
    5073 1253.69    5086 1254.54  5114.3 1262.75  5142.6 1268.46  5163.6 1270.98
  5319.4 1275.35    5379  1278.3  5439.9 1278.77  5451.1 1278.86  5471.6 1283.37
  5479.6  1283.8  5533.8 1286.63  5570.5 1289.81  5605.4 1289.33    5626 1294.65
  5654.2 1297.69  5790.6 1303.18  5811.1  1303.2  5877.5 1307.58  5909.3 1309.75
#Mann= 8 ,-1 , 0
  4693.9      .1       0  4753.4     .16       0  4998.1     .07       0
  5004.1     .16       0    5073      .1       0  5439.9     .05       0
  5479.6      .1       0  5877.5     .05       0
Bank Sta=4998.1,5004.1
XS Rating Curve= 0 ,0
Exp/Cntr=0.3,0.1

Type RM Length L Ch R = 1 ,29197   ,853,853,853
BEGIN DESCRIPTION:
CALOHAN CREEK 64.0
END DESCRIPTION:
XS GIS Cut Line= 3
      2965299.96     10043748.63      2965272.19     10044144.42
      2966014.32     10044997.53
#Sta/Elev= 30
  4421.8 1283.03  4497.1 1280.36  4513.4 1277.44  4556.1 1277.04  4707.6 1271.81
  4801.6 1270.88  4879.4 1268.05  4922.1 1262.42  4957.2 1252.03  4963.9 1247.77
  4978.1  1243.6    4997 1241.18  4999.7 1240.68    5003 1241.18  5028.5 1245.02
  5063.6 1245.06  5106.3 1247.68  5155.7 1256.92  5176.5 1263.89  5184.2 1263.92
  5190.8 1265.85  5226.9 1267.63  5268.6 1272.19    5414 1277.54  5623.8 1288.99
  5715.9 1298.77  5736.8 1302.29    5808 1308.15  5814.6 1309.87  5949.3 1315.27
#Mann= 5 ,-1 , 0
  4421.8      .1       0  4556.1     .16       0    4997     .07       0
    5003     .16       0    5414      .1       0
Bank Sta=4997,5003
XS Rating Curve= 0 ,0
Exp/Cntr=0.3,0.1

Type RM Length L Ch R = 1 ,28344   ,478,478,478
BEGIN DESCRIPTION:
CALOHAN CREEK 62.0
END DESCRIPTION:
XS GIS Cut Line= 4
      2965320.79     10043470.82      2964952.74     10044311.08
      2964862.46     10044939.56      2965385.73     10045379.66
#Sta/Elev= 30
    3695 1280.25  3789.5  1278.6  3859.6 1280.52  3917.3 1277.56  4176.7    1274
  4298.6 1272.12    4360 1268.21    4459 1266.24  4495.1 1261.72  4665.5 1254.23
  4756.5 1236.96  4785.8 1234.54    4946 1230.98  4968.6  1231.8  4995.9 1225.45
  4998.7 1224.95  5001.9 1225.45  5026.7 1233.83  5057.4 1238.43  5097.2 1247.49
  5102.3 1246.59  5120.1 1251.48  5140.4 1253.19  5243.3 1254.64  5333.1 1263.22
    5461 1268.37  5581.5 1275.15  5740.8 1280.66  5918.4 1288.78    5931 1289.87
#Mann= 10 ,-1 , 0
    3695      .1       0  4176.7     .16       0  4785.8      .1       0
    4946     .05       0  4995.9    .035       0  5001.9     .05       0
  5057.4      .1       0    5461     .16       0  5740.8      .1       0
  5918.4     .16       0
Bank Sta=4995.9,5001.9
XS Rating Curve= 0 ,0
Exp/Cntr=0.3,0.1

Type RM Length L Ch R = 1 ,27866   ,588,588,588
BEGIN DESCRIPTION:
CALOHAN CREEK 61.0
END DESCRIPTION:
XS GIS Cut Line= 4
      2964011.78     10043977.76      2964327.74     10044488.17
      2964574.27     10044984.69      2965352.02     10045390.93
#Sta/Elev= 30
  4140.1 1287.08  4140.4 1287.06  4242.7 1283.16  4362.6 1281.74  4520.4 1277.46
  4599.6 1271.88  4730.8 1271.41  4791.3 1260.09  4797.5 1256.83  4803.1  1249.9
  4819.9 1240.34  4825.5 1233.73  4842.4 1229.13  4847.9 1224.86  4892.8 1219.61
  4958.7 1221.05  4976.8 1220.74  4996.2 1217.28    4999 1216.78  5002.2 1217.28
  5021.6 1222.28  5267.6 1225.84  5333.3 1226.15  5392.6 1229.63  5406.7 1232.73
  5497.4 1248.42  5563.6 1251.65  5668.4 1263.36  5929.4 1277.64  6172.2 1288.68
#Mann= 9 ,-1 , 0
  4140.1     .16       0  4140.4      .1       0  4362.6     .16       0
  4958.7     .05       0  4996.2    .035       0  5002.2     .05       0
  5267.6      .1       0  5406.7     .16       0  5929.4      .1       0
Bank Sta=4996.2,5002.2
XS Rating Curve= 0 ,0
Exp/Cntr=0.3,0.1

Type RM Length L Ch R = 1 ,27278   ,490,490,490
BEGIN DESCRIPTION:
CALOHAN CREEK 60.0
END DESCRIPTION:
XS GIS Cut Line= 4
      2963602.07     10044408.34      2964119.41     10045179.14
      2964661.08     10045363.17      2965374.96     10045491.39
#Sta/Elev= 30
  3856.6 1289.84  4039.2 1285.37  4264.5 1279.47  4362.2 1278.49  4377.2 1275.87
  4422.7 1274.14  4542.3 1269.87  4593.3 1263.56  4826.2 1254.81  4836.7 1252.21
  4868.4 1232.73  4875.3 1226.42  4889.5 1219.82  4906.7 1215.31  4934.4 1213.63
  4997.8 1211.72  5000.6 1211.22  5003.8 1211.72  5026.8 1216.49  5189.2 1222.45
  5227.5 1226.33  5283.3 1227.13    5357  1231.3  5395.1 1235.93  5506.7 1255.42
  5547.4 1258.89  5577.9  1264.5    5638 1269.08  5974.1 1285.94  6082.3 1293.33
#Mann= 9 ,-1 , 0
  3856.6      .1       0  4039.2     .16       0  4264.5      .1       0
  4422.7     .16       0  4934.4      .1       0  4997.8     .07       0
  5003.8      .1       0  5395.1     .16       0    5638      .1       0
Bank Sta=4997.8,5003.8
XS Rating Curve= 0 ,0
Exp/Cntr=0.3,0.1

Type RM Length L Ch R = 1 ,26788   ,759,759,759
BEGIN DESCRIPTION:
CALOHAN CREEK 59.0
END DESCRIPTION:
XS GIS Cut Line= 3
      2963483.98     10045818.03      2964372.88     10045627.06
      2965369.36     10045852.74
#Sta/Elev= 30
    4292  1273.1  4351.3 1271.59  4368.6  1271.1  4439.8 1264.78  4526.7 1262.35
  4552.7 1258.42  4603.4  1255.8  4620.3 1250.64  4669.7 1247.34  4705.7 1238.66
    4714 1234.38  4719.1 1234.94  4763.4 1215.99  4807.6 1211.43  4869.4 1211.72
  4961.4 1210.97  4999.7  1205.1  5022.8 1210.79  5084.2 1211.78  5227.4 1217.78
  5268.4 1223.36  5319.7 1221.55  5350.5 1224.64    5371 1221.82  5388.1 1226.35
  5435.1 1232.85  5570.9  1257.4  5705.5 1272.44  5914.4    1281  6222.9 1301.62
#Mann= 7 ,-1 , 0
    4292     .16       0  4351.3      .1       0  4368.6     .16       0
  4552.7      .1       0  4869.4     .07       0  5084.2     .16       0
  6222.9     .05       0
Bank Sta=4869.4,5084.2
XS Rating Curve= 0 ,0
Exp/Cntr=0.3,0.1

Type RM Length L Ch R = 1 ,26029   ,388,388,388
BEGIN DESCRIPTION:
CALOHAN CREEK 57.0
END DESCRIPTION:
XS GIS Cut Line= 4
      2963459.71     10046210.39      2964001.35     10046311.08
      2964393.71      10046321.5       2964826.3     10046238.44
#Sta/Elev= 30
  4303.2 1278.49  4413.8 1271.21  4458.9  1259.9  4505.4 1241.67  4511.7 1237.79
  4565.7 1218.81  4586.7 1213.29  4622.4 1208.77  4668.1 1205.34  4698.6 1205.77
  4749.5 1202.19  4961.3 1204.79    5001 1197.66  5031.3 1203.58  5051.3 1204.48
  5061.3 1204.69  5081.3 1208.13  5091.3 1211.93  5111.3 1221.43  5139.3 1239.46
  5161.3 1248.34  5171.3 1250.13    5316 1257.17    5425  1256.5  5465.3 1254.74
  5516.2 1258.42  5567.1 1259.79  5597.7 1264.26  5638.4  1266.6  5687.1 1267.45
#Mann= 5 ,-1 , 0
  4303.2     .16       0  4565.7      .1       0  4961.3     .09       0
  5061.3     .16       0  5687.1     .05       0
Bank Sta=4961.3,5051.3
XS Rating Curve= 0 ,0
Exp/Cntr=0.3,0.1

Type RM Length L Ch R = 1 ,25641   ,485,485,485
BEGIN DESCRIPTION:
CALOHAN CREEK 56.0
END DESCRIPTION:
XS GIS Cut Line= 4
      2963456.24     10046300.68      2963796.49     10046515.94
      2964265.24     10046752.06      2964761.75     10046769.42
#Sta/Elev= 30
    4414 1276.95  4504.6 1272.88  4525.8 1270.37  4541.1 1264.03  4562.3 1259.22
  4577.5 1250.41  4598.7 1243.54    4614 1234.74  4692.8 1216.56  4708.1 1208.71
  4736.1  1202.8  4771.6  1200.1  4868.3 1197.78  4964.4 1200.35  4974.2 1198.73
  4986.8  1194.6  5001.9 1192.52  5018.8 1197.45  5031.6 1198.68  5130.4 1199.62
  5308.9 1212.29  5354.7 1213.45  5394.7 1226.64  5434.8 1236.69  5504.8 1248.23
  5564.8 1255.01  5634.9 1258.55  5674.9 1263.19  5704.9  1264.6  5838.3 1266.32
#Mann= 4 ,-1 , 0
    4414     .16       0  4974.2     .09       0  5130.4     .16       0
  5838.3      .1       0
Bank Sta=4974.2,5130.4
XS Rating Curve= 0 ,0
Exp/Cntr=0.3,0.1

Type RM Length L Ch R = 1 ,25156   ,488,488,488
BEGIN DESCRIPTION:
CALOHAN CREEK 55.0
END DESCRIPTION:
XS GIS Cut Line= 4
      2963304.29     10046482.07      2963647.19     10046933.48
      2964107.26     10047089.73      2964450.09     10047098.41
#Sta/Elev= 30
  4218.2 1278.48    4258 1275.17  4350.6 1272.38  4379.7 1266.27    4465 1260.72
  4479.5 1257.82  4550.3 1252.05  4608.5 1242.14  4643.8 1233.63  4650.1  1230.2
  4658.4 1228.78  4664.6 1223.78  4679.2  1218.6  4685.5 1213.33    4700 1207.07
  4714.6 1202.52  4749.9 1196.15    4966 1192.06  4984.9 1188.47  4990.2 1190.04
  4997.4 1186.11  5029.3 1191.84  5047.7 1194.67  5282.2 1202.53  5372.2 1211.24
  5402.2 1216.32  5452.2 1231.57  5492.2 1239.33  5542.3 1248.55  5613.9 1255.87
#Mann= 3 ,-1 , 0
  4218.2     .16       0    4966     .07       0  5029.3      .1       0
Bank Sta=4966,5029.3
XS Rating Curve= 0 ,0
Exp/Cntr=0.3,0.1

Type RM Length L Ch R = 1 ,24668   ,363,363,363
BEGIN DESCRIPTION:
CALOHAN CREEK 54.0
END DESCRIPTION:
XS GIS Cut Line= 4
      2963087.29     10046929.14      2963742.67      10047324.1
      2963985.73     10047497.72      2964314.53     10047476.08
#Sta/Elev= 30
  4028.4 1272.98  4163.6 1266.15  4258.6 1250.39  4302.5 1242.63  4338.4 1234.87
  4366.8 1224.34  4403.4 1214.17  4433.5 1213.05    4550 1199.61  4812.8 1188.99
  4854.6 1185.55  4862.2 1181.02  4875.5 1179.14  4919.7 1181.18  4925.9 1178.46
  4940.6 1178.69  4961.5 1184.84  4976.3 1184.15  4984.9  1180.3  4997.1 1176.21
  5020.5 1184.71  5034.2 1188.53  5062.3 1189.41  5082.1 1193.25  5165.2 1202.69
  5235.3 1229.32  5275.4 1239.68  5335.6 1243.21  5386.1 1249.63  5421.8 1249.87
#Mann= 7 ,-1 , 0
  4028.4     .16       0  4258.6     .05       0  4302.5      .1       0
  4366.8     .16       0  4976.3     .07       0  5082.1      .1       0
  5421.8      .1       0
Bank Sta=4984.9,5020.5
XS Rating Curve= 0 ,0
Exp/Cntr=0.3,0.1

Type RM Length L Ch R = 1 ,24305   ,363,363,363
BEGIN DESCRIPTION:
CALOHAN CREEK 53.0
END DESCRIPTION:
XS GIS Cut Line= 4
      2963039.57     10047184.36      2963451.87     10047462.13
      2963881.56     10047961.26      2964253.02     10048449.34
#Sta/Elev= 30
  4208.6 1268.59  4256.9 1266.01  4380.5 1249.34  4424.3 1239.34  4481.7 1218.36
  4514.5 1210.24  4595.7 1200.01  4768.2 1191.53  4849.9 1189.47  4938.4 1186.87
  4952.7 1184.26  4959.3 1178.92  4973.5 1174.65  4985.3  1174.6  4992.5 1174.51
  4995.2 1174.01  4998.5 1174.51  5037.7 1178.88  5262.2 1190.29  5291.1 1192.29
  5493.1 1205.56    5514 1208.29  5549.4  1221.8  5584.8 1229.82  5643.6 1236.61
  5649.2 1238.88  5692.8 1240.26  5734.5 1246.88    5828  1248.8  5977.7 1257.65
#Mann= 11 ,-1 , 0
  4208.6     .16       0  4380.5      .1       0  4514.5     .16       0
  4768.2     .05       0  4849.9     .16       0  4985.3     .05       0
  4992.5    .035       0  4998.5     .05       0  5262.2      .1       0
  5291.1     .05       0  5643.6      .1       0
Bank Sta=4992.5,4998.5
XS Rating Curve= 0 ,0
Exp/Cntr=0.3,0.1

Type RM Length L Ch R = 1 ,23942   ,421,421,421
BEGIN DESCRIPTION:
CALOHAN CREEK 52.0
END DESCRIPTION:
XS GIS Cut Line= 3
      2962922.39     10047310.25      2963547.36     10048126.19
      2963824.31     10048675.76
#Sta/Elev= 30
  4189.9 1267.02  4225.2 1266.56  4254.2  1261.8    4383 1251.52  4432.4  1240.9
  4482.7 1224.05  4509.8 1211.71  4538.9 1203.75  4576.7 1199.56  4810.9 1180.31
  4898.5 1176.52  4966.8 1174.42  4999.1 1169.71  5001.9 1169.21  5005.1 1169.71
  5008.4 1169.75  5298.4 1195.17    5343  1201.9  5359.7 1209.06  5365.3 1209.07
  5371.4 1213.57  5382.1 1218.58  5404.5 1222.56  5426.7 1228.31  5483.7 1236.92
  5566.1 1239.51  5605.1 1245.87  5665.4 1247.23  5770.1 1250.28  5833.1 1252.06
#Mann= 11 ,-1 , 0
  4189.9     .16       0  4432.4      .1       0  4576.7     .16       0
  4898.5      .1       0  4999.1     .07       0  5005.1      .1       0
  5008.4     .05       0  5371.4      .1       0  5404.5     .05       0
  5665.4      .1       0  5770.1     .05       0
Bank Sta=4999.1,5005.1
XS Rating Curve= 0 ,0
Exp/Cntr=0.3,0.1

Type RM Length L Ch R = 1 ,23521   ,463,463,463
BEGIN DESCRIPTION:
CALOHAN CREEK 51.0
END DESCRIPTION:
XS GIS Cut Line= 3
      2962627.21     10047410.02      2963126.35     10048247.72
      2963790.45     10048772.91
#Sta/Elev= 30
  4198.7 1267.34  4332.5  1263.2  4406.5 1256.14    4494 1239.49  4523.3  1240.3
  4544.7 1236.02  4560.3 1237.45  4566.1 1233.96  4581.7 1234.57  4756.9 1184.93
  4793.9 1179.99  4865.5 1176.46  4987.6 1166.42  4990.3 1165.92  4993.6 1166.42
  5087.3 1167.49  5150.2 1172.84  5165.8 1170.48  5216.7 1173.25  5257.7 1175.41
  5312.4 1183.74  5332.8 1185.86  5434.1 1194.42    5535 1204.33  5555.8 1208.93
  5599.1 1225.75  5667.9 1237.56  5706.5 1244.67  5799.2 1247.94  6020.5 1256.24
#Mann= 12 ,-1 , 0
  4198.7     .16       0  4865.5     .05       0  4987.6    .035       0
  4993.6     .05       0  5087.3      .1       0  5216.7     .05       0
  5312.4      .1       0  5332.8     .05       0  5434.1      .1       0
  5555.8     .05       0  5667.9      .1       0  5799.2     .05       0
Bank Sta=4987.6,4993.6
XS Rating Curve= 0 ,0
Exp/Cntr=0.3,0.1

Type RM Length L Ch R = 1 ,23058   ,550,550,550
BEGIN DESCRIPTION:
CALOHAN CREEK 50.0
END DESCRIPTION:
XS GIS Cut Line= 4
      2962089.03     10048217.33      2962488.33     10048460.39
      2963126.35     10048469.07      2963763.92     10048894.11
#Sta/Elev= 30
  4241.3 1249.13    4293 1244.75  4392.4 1229.17  4450.5 1211.74  4476.5 1207.58
  4699.2 1186.61  4888.9  1176.9  4968.9  1166.4  4988.9    1158  4995.9 1156.94
  4998.7 1156.44  5001.9 1156.94  5038.9 1160.49  5079.2 1160.88  5129.5 1161.89
  5228.9 1162.34  5287.9 1166.44    5309 1169.34    5318 1172.17    5329 1179.17
  5345.4 1182.38  5546.1 1197.81  5603.2 1205.22  5618.2 1208.11  5669.3 1227.84
  5756.4 1243.15  5793.6 1244.74  5857.8 1247.62  6014.8  1251.7  6113.1 1257.38
#Mann= 11 ,-1 , 0
  4241.3     .16       0    4293      .1       0  4476.5     .16       0
  4699.2      .1       0  4995.9     .07       0  5001.9      .1       0
  5079.2     .05       0  5129.5      .1       0  5287.9     .05       0
  5793.6      .1       0  5857.8     .05       0
Bank Sta=4995.9,5001.9
XS Rating Curve= 0 ,0
Exp/Cntr=0.3,0.1

Type RM Length L Ch R = 1 ,22508   ,679,679,679
BEGIN DESCRIPTION:
CALOHAN CREEK 49.0
END DESCRIPTION:
XS GIS Cut Line= 3
       2962106.4     10048668.73        2962905.     10049133.13
      2963933.53     10049055.02
#Sta/Elev= 30
  4426.6  1235.2  4563.9 1218.17  4622.7 1197.41  4783.2 1183.59  4891.7  1178.6
  4900.8  1171.4  4906.5 1170.99  4922.3 1156.78    4981 1152.23  4992.8 1148.35
  4995.6 1147.85  4998.8 1148.35  5030.5 1154.37  5107.9 1156.24  5289.5 1172.51
  5317.8 1177.95  5424.1 1183.05  5464.2 1188.94  5514.3 1202.84    5540  1205.8
    5545 1203.36  5564.5 1213.59  5604.6 1223.12  5676.2 1228.65  5905.5 1234.73
  5946.1 1240.39  6239.9  1257.6    6308 1258.68  6343.2 1260.04  6381.9 1262.91
#Mann= 9 ,-1 , 0
  4426.6      .1       0  4992.8     .07       0  4998.8      .1       0
  5107.9     .05       0  5289.5      .1       0  5946.1     .05       0
  6239.9      .1       0    6308     .05       0  6343.2      .1       0
Bank Sta=4992.8,4998.8
XS Rating Curve= 0 ,0
Exp/Cntr=0.3,0.1

Type RM Length L Ch R = 1 ,21829   ,703,703,703
BEGIN DESCRIPTION:
CALOHAN CREEK 47.0
END DESCRIPTION:
XS GIS Cut Line= 2
      2962006.53     10048963.83      2963377.95     10050278.83
#Sta/Elev= 30
  4144.4 1232.07    4181 1225.72  4209.3 1216.63  4223.5 1206.39  4280.1  1192.7
  4541.8 1168.76  4693.6 1161.43  4915.6 1149.62  4956.2 1146.64  4991.3 1140.39
  4994.1 1139.89  4997.3 1140.39  5050.9 1142.28  5079.2 1155.77  5107.5 1173.99
  5125.8 1176.44  5229.9 1180.66  5333.9 1185.83  5461.3 1197.28  5475.5 1199.05
  5510.7 1211.92  5524.8 1215.13  5553.1 1219.88  5581.4 1221.51  5588.1 1224.08
  5673.3 1235.41  5729.9 1240.52  5839.8 1244.64  5885.6 1249.48  6044.4 1252.91
#Mann= 10 ,-1 , 0
  4144.4      .1       0  4693.6     .05       0  4915.6      .1       0
  4956.2     .05       0  4991.3    .035       0  4997.3     .05       0
  5125.8      .1       0  5229.9     .05       0  5588.1      .1       0
  5839.8     .05       0
Bank Sta=4991.3,4997.3
XS Rating Curve= 0 ,0
Exp/Cntr=0.3,0.1

Type RM Length L Ch R = 1 ,21126   ,266,266,266
BEGIN DESCRIPTION:
CALOHAN CREEK 46.0
END DESCRIPTION:
XS GIS Cut Line= 4
      2961893.71     10048989.86      2961963.16     10049454.31
      2961984.86     10049771.15      2962792.19     10050265.97
#Sta/Elev= 30
  4340.5 1240.37  4403.2 1239.45  4506.2 1230.41  4526.4 1223.94  4541.6 1213.35
  4587.1 1196.85  4627.5 1188.56    4675 1165.88  4728.2 1147.94  4779.2 1141.51
  4851.8 1140.46  4917.3 1139.89 4973.86 1135.94    4997 1130.71  4999.7 1130.21
    5003 1130.71  5070.1 1135.97  5124.7 1136.96  5133.7  1136.9  5300.7 1138.05
  5372.1 1147.29  5408.8 1158.08  5430.1  1159.8  5466.9 1172.51  5584.8 1177.77
  5882.6 1196.17  5931.1    1204  5983.2 1219.21  6041.3 1228.68  6074.6 1229.62
#Mann= 10 ,-1 , 0
  4340.5     .16       0  4728.2      .1       0  4851.8     .05       0
  4917.3      .1       0    4997     .07       0    5003      .1       0
  5124.7     .05       0  5133.7      .1       0  5300.7     .16       0
  5584.8      .1       0
#XS Ineff= 3 ,-1
 5176.94 5230.96  1136.8  5271.4 5284.48 1137.58  5293.6 5305.44 1138.43
Permanent Ineff=
       T       T       T
Bank Sta=4973.86,5070.1
XS Rating Curve= 0 ,0
Exp/Cntr=0.3,0.1

Type RM Length L Ch R = 1 ,20860   ,356,356,356
BEGIN DESCRIPTION:
CALOHAN CREEK 45.0
END DESCRIPTION:
XS GIS Cut Line= 3
      2961533.48     10049536.78       2961945.8     10049918.72
      2962770.47     10050305.02
#Sta/Elev= 30
  4678.9 1179.56  4854.6 1174.56  4878.2  1170.2  4885.6 1161.84  4892.4 1161.47
  4902.6 1155.45  4920.7 1148.74  4928.1 1134.03  4942.3 1129.89    4996 1127.99
  4998.7 1127.49    5002 1127.99  5019.9  1133.5    5032 1133.79  5282.1 1133.31
  5482.5 1135.92  5524.7 1141.54    5542 1149.39  5547.5    1148  5570.3 1157.69
  5575.8 1156.36  5593.2 1164.08  5598.7 1162.52  5611.2 1167.52  5638.8 1173.92
  5855.3 1186.02    5975 1196.38  5997.8 1201.03    6050 1218.35  6151.6 1229.41
#Mann= 9 ,-1 , 0
  4678.9      .1       0  4854.6     .16       0  4902.6      .1       0
    4996     .07       0    5002      .1       0    5032     .05       0
  5282.1      .1       0  5482.5     .16       0  5611.2      .1       0
#XS Ineff= 3 ,-1
  5026.5 5088.38 1133.96 5090.94 5101.78 1134.56 5104.34  6151.6  1134.9
Permanent Ineff=
       T       T       T
Bank Sta=4928.1,5019.9
XS Rating Curve= 0 ,0
Exp/Cntr=0.3,0.1

Type RM Length L Ch R = 1 ,20504   ,461,461,461
BEGIN DESCRIPTION:
Mapping XS 525c2f8d
END DESCRIPTION:
XS GIS Cut Line= 4
      2961519.32     10049678.22      2961857.88     10050053.24
      2961970.73     10050051.51      2962713.62     10050325.75
#Sta/Elev= 30
  4445.8 1175.91  4700.5 1171.47  4781.8  1154.7  4841.2 1150.16    4867 1148.96
  4873.7 1143.97  4881.2 1147.38  4887.9 1141.17  4895.4 1144.29  4902.1 1138.28
  4909.6 1141.63  4916.3  1135.8  4923.8 1138.93  4944.7 1130.73  4953.8 1133.49
  4971.6 1124.83  4972.6 1124.69  4998.6 1122.46  5001.4 1121.96  5004.6 1122.46
  5031.6 1126.28  5071.7 1126.97  5278.8 1136.65    5328 1140.98  5367.7 1154.78
  5423.9 1174.33  5701.1 1193.08    5749 1201.18  5804.5 1218.54  5855.8 1224.78
#Mann= 9 ,-1 , 0
  4445.8     .16       0  4700.5      .1       0  4841.2     .05       0
  4972.6     .16       0  4998.6     .07       0  5004.6     .16       0
  5071.7      .1       0  5278.8     .16       0  5367.7      .1       0
Bank Sta=4971.6,5031.6
XS Rating Curve= 0 ,0
Exp/Cntr=0.3,0.1

Type RM Length L Ch R = 1 ,20043   ,399,399,399
BEGIN DESCRIPTION:
CALOHAN CREEK 43.0
END DESCRIPTION:
XS GIS Cut Line= 4
      2961589.91     10049862.32      2961863.33     10050352.75
      2962306.04      10050574.1      2962818.17     10050660.91
#Sta/Elev= 30
  4217.2 1173.34  4408.7  1164.6  4433.2 1162.57  4533.1 1152.62  4549.1 1146.71
  4596.9 1141.44  4673.7 1128.62  4717.1 1125.26  4776.4 1122.57  4858.1  1124.4
  4985.7 1119.74  4992.2 1116.47  4994.9 1115.31  4997.6 1114.81  5000.9 1115.31
    5037  1121.8  5052.8 1124.63  5075.1 1134.31  5087.3 1145.17  5094.8 1148.38
  5119.9 1157.11  5154.4 1176.52  5327.9 1187.75  5422.1 1196.66  5458.7 1211.33
  5474.2 1213.47  5509.4  1219.2  5663.5 1230.61    5692  1236.5  5793.1 1243.07
#Mann= 10 ,-1 , 0
  4217.2     .16       0  4408.7      .1       0  4433.2     .16       0
  4596.9      .1       0  4992.2     .16       0  4994.9     .07       0
  5000.9     .16       0  5094.8      .1       0  5327.9     .16       0
  5474.2      .1       0
#XS Ineff= 2 ,-1
  4217.2 4857.86 1124.46 4885.95 4925.11 1122.56
Permanent Ineff=
       T       T
Bank Sta=4985.7,5037
XS Rating Curve= 0 ,0
Exp/Cntr=0.3,0.1

Type RM Length L Ch R = 1 ,19644   ,1123,1123,1123
BEGIN DESCRIPTION:
CALOHAN CREEK 42.0
END DESCRIPTION:
XS GIS Cut Line= 2
      2960201.01     10050157.44      2962934.46     10050977.47
#Sta/Elev= 30
  3403.8 1232.93  3511.7 1226.06  3589.1  1205.5  3813.4 1191.04  4288.6 1166.91
  4361.6 1153.34  4417.6 1127.88  4554.5 1118.14    4591 1110.35  4593.8 1109.85
    4597 1110.35  4676.6 1115.77  4926.1 1117.11  4973.4 1118.12  5006.4 1111.46
  5110.8 1119.73  5116.1 1126.44  5129.5 1131.19  5143.9 1134.53  5149.1 1144.24
  5231.2 1165.95    5333 1176.44    5488 1184.65  5638.1 1193.25  5742.5 1200.49
  5813.8 1215.72  5874.7 1219.79    5959 1235.56  6044.9 1241.81  6257.6  1256.6
#Mann= 14 ,-1 , 0
  3403.8      .1       0  3813.4     .16       0  4417.6      .1       0
  4554.5     .16       0    4591     .07       0    4597     .16       0
  4676.6     .05       0  4926.1     .16       0  5129.5      .1       0
  5231.2     .16       0    5333      .1       0    5488     .16       0
  5638.1     .05       0  6044.9      .1       0
#XS Ineff= 2 , 0
         4972.51 1118.12
Permanent Ineff=
       T       T
Bank Sta=4973.4,5110.8
XS Rating Curve= 0 ,0
Exp/Cntr=0.3,0.1

Type RM Length L Ch R = 1 ,18521   ,607,607,607
BEGIN DESCRIPTION:
CALOHAN CREEK 40.0
END DESCRIPTION:
XS GIS Cut Line= 4
      2959897.18     10051016.81      2960817.33     10051151.36
      2962023.92     10051581.05      2962755.49     10051645.98
#Sta/Elev= 30
  3786.8 1232.34  3872.6 1224.16  3927.8 1213.13  4006.4 1204.12  4058.9 1202.34
  4682.1 1179.02  4741.6 1176.73  4859.6 1163.58  4890.4 1152.85  4915.9 1132.15
  4921.2 1132.57  4946.8 1113.53  4953.3 1112.25  4972.3  1103.3  4990.9 1100.67
  4993.7 1100.17  4996.9 1100.67  5033.9  1105.6  5078.9 1104.35  5497.7 1123.19
  5547.4 1126.73  5603.7 1136.39  5665.4 1149.32  5690.9  1158.2  5870.6 1173.69
  6314.5 1194.73  6373.6 1201.89  6421.3 1220.29    6484 1229.89    6732 1243.13
#Mann= 9 ,-1 , 0
  3786.8     .05       0  3872.6      .1       0  3927.8     .05       0
  4058.9      .1       0  4682.1     .16       0  4953.3     .05       0
  4990.9    .035       0  4996.9     .05       0  5497.7      .1       0
Bank Sta=4990.9,4996.9
XS Rating Curve= 0 ,0
Exp/Cntr=0.3,0.1

Type RM Length L Ch R = 1 ,17914   ,618,618,618
BEGIN DESCRIPTION:
CALOHAN CREEK 38.0
END DESCRIPTION:
XS GIS Cut Line= 4
      2959819.06     10051160.04      2960552.57     10051528.97
      2961416.28     10052080.18      2962510.05     10052410.05
#Sta/Elev= 30
  3642.2 1238.44    3678 1237.74  3902.5 1213.63  4319.7 1188.71  4572.7 1179.02
  4651.4  1169.9  4724.2 1151.24  4739.4 1140.36    4797  1114.7  4839.3 1105.16
  4897.8 1100.74  4949.3  1100.5    4997 1092.54  4999.8 1092.04    5003 1092.54
    5004 1092.67  5125.7 1101.36  5145.1 1102.71  5246.7 1106.03  5397.3 1108.51
  5467.6 1109.82  5636.4 1115.99  5673.3 1121.69  5834.8 1156.76  5978.5 1165.44
    5983 1165.69  6075.5 1172.13  6365.7 1176.87  6510.5  1180.1  6630.3 1185.38
#Mann= 20 ,-1 , 0
  3642.2      .1       0    3678     .05       0  3902.5      .1       0
  4319.7     .16       0  4897.8      .1       0  4949.3     .16       0
    4997     .07       0    5003     .16       0    5004      .1       0
  5125.7     .05       0  5145.1      .1       0  5246.7     .05       0
  5397.3      .1       0  5467.6     .16       0  5673.3      .1       0
  5978.5     .05       0    5983     .16       0  6075.5      .1       0
  6365.7     .05       0  6510.5      .1       0
Bank Sta=4997,5003
XS Rating Curve= 0 ,0
Exp/Cntr=0.3,0.1

Type RM Length L Ch R = 1 ,17296   ,996,996,996
BEGIN DESCRIPTION:
CALOHAN CREEK 37.0
END DESCRIPTION:
XS GIS Cut Line= 4
      2960031.69     10052318.89      2960565.59     10052444.76
      2961290.42     10052314.56      2962510.07     10052783.32
#Sta/Elev= 30
  4071.7 1225.37  4114.6 1219.07  4142.4 1206.34  4181.4  1197.5  4511.1 1178.75
  4633.3 1160.94  4710.2 1136.61    4829 1117.16  4907.6  1110.7  4948.3  1093.3
  4996.1 1085.62  4998.8 1085.12  5002.1 1085.62  5039.7 1093.73  5133.2 1094.36
  5280.7 1096.25  5326.9 1097.64  5460.3 1101.16  5564.3  1106.3    5607 1109.06
  5668.3 1114.03  5787.4 1131.51  5879.5 1156.49    5934 1163.82  5981.4 1174.06
  6254.5 1188.01    6308  1196.7  6326.7 1205.35  6430.7 1226.45  6663.3 1230.35
#Mann= 15 ,-1 , 0
  4071.7     .05       0  4142.4      .1       0    4829     .16       0
  4996.1     .07       0  5002.1     .16       0  5133.2      .1       0
  5280.7     .05       0  5326.9      .1       0  5460.3     .05       0
  5564.3     .16       0    5607     .05       0  5668.3     .16       0
    5934      .1       0  6326.7     .05       0  6430.7      .1       0
Bank Sta=4996.1,5002.1
XS Rating Curve= 0 ,0
Exp/Cntr=0.3,0.1

Type RM Length L Ch R = 1 ,16300   ,469,469,469
BEGIN DESCRIPTION:
CALOHAN CREEK 35.0
END DESCRIPTION:
XS GIS Cut Line= 4
      2960109.88     10052570.64      2960995.28     10053095.81
      2961273.06      10053343.2      2961980.51     10053460.39
#Sta/Elev= 30
  3784.4 1195.15  3802.6 1193.89  4143.2 1177.48  4201.3 1170.12  4353.7  1159.9
  4378.7 1152.48  4412.2 1141.47    4422 1141.45  4427.8 1136.97  4480.4 1128.68
  4571.6 1107.74  4692.6 1096.11  4868.3 1085.87  4963.6  1086.5  5024.1 1082.87
  5030.9 1082.55  5033.6 1082.05  5036.9 1082.55    5183 1109.55  5230.8 1121.52
  5284.2 1135.26  5340.1 1154.62  5357.6 1157.02  5424.4 1171.85  5456.9 1174.24
  5667.7 1188.31  5711.2 1197.36  5754.9 1215.08  5809.6 1227.25  5902.9 1233.43
#Mann= 14 ,-1 , 0
  3784.4     .05       0  3802.6      .1       0  4378.7     .16       0
  4571.6      .1       0  4692.6     .05       0  4868.3      .1       0
  5024.1     .16       0  5030.9     .07       0  5036.9     .16       0
    5183      .1       0  5230.8     .16       0  5357.6      .1       0
  5456.9     .05       0  5754.9     .16       0
Bank Sta=5030.9,5036.9
XS Rating Curve= 0 ,0
Exp/Cntr=0.3,0.1

Type RM Length L Ch R = 1 ,15831   ,351,351,351
BEGIN DESCRIPTION:
CALOHAN CREEK 34.0
END DESCRIPTION:
XS GIS Cut Line= 4
      2959931.89     10052679.11      2960622.01     10053577.58
      2961550.83     10053638.34      2962050.01     10053551.53
#Sta/Elev= 30
  3430.3 1190.94  3765.7 1178.28    3809 1173.66  3984.3 1167.63  4137.7 1162.19
  4266.3 1159.39  4315.9 1157.49  4394.5 1146.84  4541.3 1120.67  4585.7 1115.22
  4671.9 1099.42    4700 1093.69  4851.3    1091  4920.4 1088.92  4977.6 1082.28
  4980.3 1081.78  4983.6 1082.28  5078.7  1087.1  5194.8 1095.06  5291.2 1107.54
  5341.3 1120.12  5421.5 1152.16  5473.1 1167.54  5490.3 1173.83  5573.5 1178.47
  5714.9 1191.72  5727.7 1194.43  5775.3 1216.08  5836.7 1227.97  6000.7 1235.34
#Mann= 16 ,-1 , 0
  3430.3      .1       0    3809     .05       0  3984.3      .1       0
  4137.7     .16       0  4266.3     .05       0  4394.5      .1       0
  4541.3     .05       0  4585.7      .1       0  4671.9     .05       0
  4851.3      .1       0  4977.6     .07       0  4983.6      .1       0
  5078.7     .16       0  5473.1      .1       0  5573.5     .05       0
  5775.3     .16       0
Bank Sta=4977.6,4983.6
XS Rating Curve= 0 ,0
Exp/Cntr=0.3,0.1

Type RM Length L Ch R = 1 ,15480   ,572,572,572
BEGIN DESCRIPTION:
CALOHAN CREEK 33.0
END DESCRIPTION:
XS GIS Cut Line= 2
      2959720.95     10053923.93      2961950.14     10053930.88
#Sta/Elev= 30
    3682 1168.05  3745.8 1166.13  3949.5 1160.79    4043 1148.81  4053.4 1146.92
  4129.5 1131.58  4379.5 1107.04  4509.5  1099.7  4570.1 1090.78  4590.7 1088.87
  4689.4 1085.13  4889.5 1081.72  4936.5  1077.8  4939.3  1077.3  4942.5  1077.8
  5049.5  1078.6  5119.5 1085.72  5149.5 1091.58  5223.9 1094.77  5299.5 1102.93
  5389.5 1131.28  5419.5 1146.44  5469.5 1159.05  5509.5 1173.78  5608.9 1179.23
  5729.5  1188.5  5749.5 1192.05  5774.5 1200.97  5819.5 1216.56  5911.2 1225.64
#Mann= 11 ,-1 , 0
    3682     .16       0  3745.8      .1       0    4043     .05       0
  4053.4      .1       0  4570.1     .05       0  4590.7      .1       0
  4689.4     .16       0  4936.5     .07       0  4942.5     .16       0
  5608.9      .1       0  5774.5     .16       0
Bank Sta=4936.5,4942.5
XS Rating Curve= 0 ,0
Exp/Cntr=0.3,0.1

Type RM Length L Ch R = 1 ,15184   ,89,89,89
BEGIN DESCRIPTION:
CALOHAN CREEK 67.0
END DESCRIPTION:
XS GIS Cut Line= 4
      2959561.37     10053940.78      2960686.32     10054173.41
       2961401.6     10054208.13      2961721.02     10054267.15
#Sta/Elev= 30
  3423.8 1174.69  3540.1 1170.31  3956.9 1160.33    4002 1155.16    4007 1156.32
  4092.8 1142.92  4152.7 1132.99    4208  1130.7  4298.2 1119.74  4361.2 1117.28
  4404.7 1114.82  4504.6 1106.73  4576.1 1098.27  4604.7 1089.97  4636.2 1085.71
  4744.9 1078.58    4822 1077.28  4824.7 1076.78    4828 1077.28  4998.4 1078.42
  5065.3 1078.97  5115.3 1089.18  5145.4 1100.05  5185.4 1118.32  5195.4 1123.85
  5225.5 1146.84  5291.3 1170.91  5513.2 1181.07  5592.8 1186.97  5613.5 1188.26
#Mann= 12 ,-1 , 0
  3423.8     .16       0  3540.1      .1       0    4007     .05       0
  4092.8      .1       0  4361.2     .05       0  4404.7      .1       0
  4504.6     .16       0  4636.2     .05       0    4822     .07       0
    4828     .05       0  4998.4     .16       0  5592.8      .1       0
Bank Sta=4822,4828
XS Rating Curve= 0 ,0
Exp/Cntr=0.3,0.1

Type RM Length L Ch R = 1 ,15095   ,187,187,187
BEGIN DESCRIPTION:
CALOHAN CREEK 66.0
END DESCRIPTION:
XS GIS Cut Line= 6
      2959533.51     10053972.01       2960776.6     10054294.93
      2961037.71     10054297.25      2961148.82     10054278.15
      2961523.82     10054376.24      2961763.32     10054432.31
#Sta/Elev= 30
  3366.1 1178.04  3414.9 1176.35  3470.9 1172.19  3683.6 1167.94  3803.2 1164.53
  3992.9 1160.13    4081 1148.62  4144.7 1138.41  4149.9 1140.26  4177.1 1133.15
    4231 1128.86  4266.4 1122.68  4383.5 1114.01  4482.3  1105.2  4545.1  1094.2
  4593.7 1089.16  4799.3 1074.79  4802.1 1074.29  4805.3 1074.79  4892.3 1077.06
  4909.7 1079.83  5034.3 1081.44  5068.3 1077.48    5117 1102.03    5179 1126.59
  5184.4 1133.57  5199.7 1144.76  5230.7 1163.12  5251.3 1170.06  5657.9  1187.2
#Mann= 11 ,-1 , 0
  3366.1     .16       0  3414.9      .1       0  3683.6     .05       0
  3803.2      .1       0    4081     .05       0  4383.5      .1       0
  4482.3     .16       0  4593.7     .05       0  4799.3     .07       0
  4805.3     .05       0  4909.7     .16       0
Bank Sta=4799.3,4805.3
XS Rating Curve= 0 ,0
Exp/Cntr=0.3,0.1

Type RM Length L Ch R = 1 ,14908   ,484,484,484
BEGIN DESCRIPTION:
CALOHAN CREEK 32.0
END DESCRIPTION:
XS GIS Cut Line= 4
      2959514.36      10054033.3      2960493.54     10054265.08
      2961418.02     10054561.95      2961699.26     10054567.16
#Sta/Elev= 30
  3336.2  1182.2  3340.3  1182.2    3583 1171.23  3890.3  1162.6  4012.3 1158.95
  4064.8 1151.34  4144.2 1142.46  4181.3 1132.99  4186.4 1133.95  4366.4 1110.82
  4460.9 1103.71  4514.2 1095.51  4592.2 1089.13  4749.4  1078.5  4820.2 1070.61
  4841.5 1071.63  4872.6 1074.33  4956.8 1074.34  4988.3 1065.59  5003.3 1065.02
    5006 1064.52  5009.3 1065.02  5051.3 1096.68  5082.8 1114.17  5107.9 1122.52
  5134.7  1134.6    5140 1134.14  5166.8 1148.34  5261.4 1169.37  5594.7 1180.31
#Mann= 11 ,-1 , 0
  3336.2     .05       0  3340.3      .1       0    3583     .05       0
  3890.3      .1       0  4064.8     .05       0  4366.4      .1       0
  4460.9     .16       0  4592.2     .05       0  4841.5     .16       0
  5003.3     .07       0  5009.3     .16       0
Bank Sta=5003.3,5009.3
XS Rating Curve= 0 ,0
Exp/Cntr=0.3,0.1

Type RM Length L Ch R = 1 ,14424   ,923,923,923
BEGIN DESCRIPTION:
CALOHAN CREEK 31.0
END DESCRIPTION:
XS GIS Cut Line= 4
      2959929.48      10054472.3      2960590.98     10054810.87
       2961288.9     10055013.99      2961704.49      10054899.7
#Sta/Elev= 30
  3885.2 1164.73  3921.7 1163.63  3965.2 1162.31    4100  1159.9  4149.8 1150.81
  4221.1 1142.15  4249.8 1130.43  4299.9 1126.76  4421.9 1111.04  4491.4 1106.19
  4577.3  1098.8  4614.2 1089.94  4719.4  1082.3    4780 1072.69  4783.2 1072.31
  4886.1 1063.18  4917.3 1068.01  4937.8 1067.95  4976.6 1061.51  4997.6 1061.38
  5000.4 1060.88  5003.6 1061.38  5031.9 1064.18  5082.3 1078.96    5232 1106.62
    5299 1126.29  5337.7 1132.21  5412.3 1154.75  5645.1 1168.08  5786.2 1169.72
#Mann= 9 ,-1 , 0
  3885.2     .16       0  3921.7      .1       0  3965.2     .16       0
  4149.8      .1       0  4491.4     .16       0    4780      .1       0
  4783.2     .16       0  4997.6     .07       0  5003.6     .16       0
Bank Sta=4997.6,5003.6
XS Rating Curve= 0 ,0
Exp/Cntr=0.3,0.1

Type RM Length L Ch R = 1 ,13501   ,649,649,649
BEGIN DESCRIPTION:
CALOHAN CREEK 29.0
END DESCRIPTION:
XS GIS Cut Line= 4
      2959710.77     10055404.62      2960804.52      10055831.7
      2961273.27     10055717.12      2961611.52     10055368.46
#Sta/Elev= 30
  3618.7    1168  3619.2 1167.97  3786.1 1163.46  3820.2 1162.54    3873 1154.63
  3992.4 1143.15  4057.4 1132.32  4125.5  1123.7    4150 1116.89  4271.1  1107.2
  4314.4 1099.55  4550.2 1076.34    4627 1072.75  4920.5 1060.43  4951.4 1057.07
  4989.5 1047.88  4992.3 1047.38  4995.5 1047.88  5020.7 1050.47  5033.7  1048.8
  5058.8 1056.18  5126.4 1059.52  5136.7 1061.72  5208.7 1096.81    5338 1112.18
  5444.2 1130.38  5571.5 1141.69  5635.1 1144.21  5663.4 1149.28  5761.2  1151.7
#Mann= 10 ,-1 , 0
  3618.7      .1       0  3619.2     .05       0  3786.1      .1       0
  3820.2     .05       0  4057.4      .1       0  4314.4     .16       0
    4627      .1       0  4989.5     .07       0  4995.5      .1       0
  5020.7     .16       0
Bank Sta=4989.5,4995.5
XS Rating Curve= 0 ,0
Exp/Cntr=0.3,0.1

Type RM Length L Ch R = 1 ,12852   ,483,483,483
BEGIN DESCRIPTION:
CALOHAN CREEK 28.0
END DESCRIPTION:
XS GIS Cut Line= 4
      2959622.21     10055420.23      2960861.81     10056336.91
      2961346.19     10056493.16      2962533.53     10056513.99
#Sta/Elev= 30
  3284.1 1169.37  3563.4 1162.77  3589.6 1157.89  3713.1 1149.55  3733.6  1148.1
  3890.5 1132.08  4019.9 1116.14  4106.1 1107.54  4170.8 1093.25  4423.9  1070.9
    4601 1064.13  4825.8 1057.09  4948.2 1047.27  4992.2 1039.18  4994.9 1038.68
  4998.2 1039.18  5021.9 1042.08  5059.2 1058.47  5092.7 1061.12  5096.1 1061.07
    5195 1066.08  5364.5 1075.93  5495.8 1086.82  5594.4 1095.98  5717.1 1109.38
  5937.1  1148.6    6186 1161.07  6300.2  1167.6  6368.4 1170.09  6522.3 1175.46
#Mann= 20 ,-1 , 0
  3284.1      .1       0  3589.6     .05       0  3713.1      .1       0
  3733.6     .16       0  3890.5      .1       0  4019.9     .05       0
  4423.9      .1       0    4601     .05       0  4948.2      .1       0
  4992.2     .07       0  4998.2      .1       0  5092.7     .05       0
  5096.1      .1       0    5195     .16       0  5364.5      .1       0
  5495.8     .16       0  5594.4     .05       0    6186      .1       0
  6300.2     .05       0  6368.4      .1       0
Bank Sta=4992.2,4998.2
XS Rating Curve= 0 ,0
Exp/Cntr=0.3,0.1

Type RM Length L Ch R = 1 ,12369   ,592,592,592
BEGIN DESCRIPTION:
CALOHAN CREEK 26.0
END DESCRIPTION:
XS GIS Cut Line= 3
      2959846.22     10057019.19      2960669.11      10056831.7
      2962257.61     10056998.36
#Sta/Elev= 30
  3853.4 1161.78  3927.5 1160.87  3987.2 1151.49  4153.1 1138.87  4169.5 1134.75
  4260.7 1125.02  4303.7 1117.19  4542.9 1101.39  4583.9 1089.31  4635.2    1081
  4686.5 1062.56  4731.9 1057.97  4887.8 1050.01  5005.4 1036.89  5008.2 1036.39
  5011.4 1036.89  5046.3 1041.21  5110.7 1050.24  5244.3 1058.95    5300 1065.24
  5350.3 1074.75  5430.7 1079.53    5659 1107.37  5680.9 1114.09  5792.7 1140.02
  5818.3 1150.36  5883.2 1155.03  5963.7 1165.54  6170.8 1174.82  6294.6 1181.16
#Mann= 10 ,-1 , 0
  3853.4     .16       0  4731.9     .05       0  5005.4    .035       0
  5011.4     .05       0  5046.3      .1       0  5110.7     .16       0
    5659      .1       0  5680.9     .16       0  5818.3      .1       0
  6170.8     .05       0
Bank Sta=5005.4,5011.4
XS Rating Curve= 0 ,0
Exp/Cntr=0.3,0.1

Type RM Length L Ch R = 1 ,11777   ,833,833,833
BEGIN DESCRIPTION:
CALOHAN CREEK 25.0
END DESCRIPTION:
XS GIS Cut Line= 3
      2959992.05     10057217.12      2961637.86     10057638.99
      2961934.14     10057638.99
#Sta/Elev= 30
  4158.1 1160.45    4366 1140.28  4505.4 1114.21    4588 1104.57  4610.7 1099.46
  4634.5 1098.88  4660.2  1090.2  4722.2 1078.96    4733 1072.66  4768.7 1060.18
    4868 1048.77  4931.8 1043.73  4997.9 1029.57  5000.7 1029.07  5003.9 1029.57
  5069.5 1040.21  5130.5 1047.09  5223.8 1050.24  5375.3 1052.53    5393 1055.74
    5416  1059.4  5475.8 1076.19  5517.1 1082.57  5558.4 1094.97  5635.5 1102.24
  5777.9 1123.08  5877.7 1141.39  5907.7 1150.04  6039.4 1159.35  6153.4 1168.68
#Mann= 10 ,-1 , 0
  4158.1     .16       0  4634.5      .1       0    4868     .05       0
  4997.9    .035       0  5003.9     .05       0  5069.5     .16       0
  5223.8      .1       0    5393     .16       0  5635.5      .1       0
  6039.4     .16       0
Bank Sta=4997.9,5003.9
XS Rating Curve= 0 ,0
Exp/Cntr=0.3,0.1

Type RM Length L Ch R = 1 ,10944   ,705,705,705
BEGIN DESCRIPTION:
CALOHAN CREEK 24.0
END DESCRIPTION:
XS GIS Cut Line= 3
      2960018.08     10057540.04      2960960.77     10058008.78
      2961974.94     10057712.33
#Sta/Elev= 30
  3616.9 1160.92  3639.1 1160.06  3760.9 1145.47  3829.5 1138.57  3876.2 1129.53
  3948.8  1117.1    4044 1107.04  4115.9 1085.09  4231.6 1058.98  4312.6 1054.27
  4334.4 1053.12  4603.9 1045.59  4752.3 1037.18    4921 1035.54  4957.9 1029.41
  4997.7 1023.78  5000.4 1023.28  5003.7 1023.78  5026.5 1024.59  5065.2  1032.6
  5093.4 1049.97  5098.6 1048.96  5104.9 1058.14  5165.5 1092.75  5209.6 1102.73
    5282 1119.49  5438.3 1142.24  5469.5 1150.58  5536.7 1154.79  5726.3 1168.93
#Mann= 13 ,-1 , 0
  3616.9     .16       0  3639.1      .1       0  3760.9     .16       0
  3876.2      .1       0  4115.9     .05       0  4312.6      .1       0
  4334.4     .05       0  4752.3      .1       0  4957.9     .16       0
  4997.7     .07       0  5003.7     .16       0  5209.6      .1       0
  5536.7     .16       0
Bank Sta=4997.7,5003.7
XS Rating Curve= 0 ,0
Exp/Cntr=0.3,0.1

Type RM Length L Ch R = 1 ,10239   ,393,393,393
BEGIN DESCRIPTION:
CALOHAN CREEK 22.0
END DESCRIPTION:
XS GIS Cut Line= 4
      2960023.24     10057592.09      2960590.98     10058107.74
      2960955.56     10058607.74      2961735.12       10058852.
#Sta/Elev= 30
  3906.6 1160.25    3961 1151.62  4032.1 1145.44  4102.8 1139.71  4150.8  1131.5
  4364.5 1105.54  4378.6 1102.51  4395.5 1093.63  4421.2 1082.83  4492.9 1066.41
  4555.7  1055.4  4750.4 1044.71  4759.3 1044.39  4995.4 1022.57  4998.2 1022.07
  5001.4 1022.57  5219.8 1042.97    5285 1049.31  5361.9 1068.33  5379.2 1076.06
  5421.2 1083.34  5442.1 1091.56  5473.6 1097.75  5668.1 1109.14    5746 1115.18
  5795.3 1123.88  5924.6 1137.71  6032.8 1144.86  6049.9 1149.73  6109.3 1151.35
#Mann= 13 ,-1 , 0
  3906.6      .1       0  4032.1     .16       0  4150.8      .1       0
  4395.5     .05       0  4492.9      .1       0  4750.4     .05       0
  4759.3      .1       0  4995.4     .07       0  5001.4      .1       0
  5219.8      .1       0  5361.9     .16       0  5668.1      .1       0
  5924.6     .05       0
Bank Sta=4995.4,5001.4
XS Rating Curve= 0 ,0
Exp/Cntr=0.3,0.1

Type RM Length L Ch R = 1 ,9846    ,397,397,397
BEGIN DESCRIPTION:
CALOHAN CREEK 21.0
END DESCRIPTION:
XS GIS Cut Line= 4
      2959424.34     10058347.33      2960132.65     10058441.07
      2960835.77     10058826.49      2961663.67     10058925.42
#Sta/Elev= 30
  3847.6 1165.29  3952.6 1162.46  4009.4 1153.67  4154.4 1140.89  4282.2 1120.29
  4351.1 1111.07  4396.7 1106.14  4517.5 1073.86    4628 1057.85  4720.7 1049.86
    4945 1034.05  4973.4 1024.27  4979.3 1016.57  4986.5 1015.21  4989.3 1014.71
  4992.5 1015.21  5011.3  1015.7  5012.2 1015.79  5104.7 1028.62  5136.5 1027.39
  5245.5 1037.18  5342.1 1061.71  5396.8 1077.98  5443.2 1083.04  5517.7 1087.93
  5578.1 1097.94  5838.6 1111.32  6031.5 1130.92  6112.1 1138.74  6197.7 1143.26
#Mann= 14 ,-1 , 0
  3847.6      .1       0  4282.2     .16       0  4351.1      .1       0
    4628     .16       0  4720.7     .05       0  4986.5    .035       0
  4992.5     .05       0  5011.3      .1       0  5012.2     .05       0
  5342.1      .1       0  5443.2     .16       0  5838.6      .1       0
  6031.5     .05       0  6112.1      .1       0
Bank Sta=4986.5,4992.5
XS Rating Curve= 0 ,0
Exp/Cntr=0.3,0.1

Type RM Length L Ch R = 1 ,9449    ,680,680,680
BEGIN DESCRIPTION:
CALOHAN CREEK 20.0
END DESCRIPTION:
XS GIS Cut Line= 3
      2959330.58     10058472.33       2960476.4     10059076.49
      2961673.85     10059060.87
#Sta/Elev= 30
  3857.8 1166.43  3979.5 1163.79  4064.5 1161.71  4156.2 1149.57  4228.5  1142.5
  4420.7 1106.64  4449.7 1093.54  4488.1 1084.41  4535.3  1063.7  4576.2 1049.96
  4620.2 1042.29  4889.2 1030.51  4971.7 1024.54  4994.2 1013.44    4997 1012.94
  5000.2 1013.44  5080.8 1022.94  5087.4 1023.83  5186.4 1028.62  5245.2 1045.32
  5285.1  1050.1  5383.8 1059.41  5482.6 1064.46  5615.3 1081.59  5662.4 1083.41
  5744.2 1087.71  5825.3 1098.25  5976.2 1105.59  6255.3 1130.39  6350.7 1133.46
#Mann= 16 ,-1 , 0
  3857.8     .16       0  3979.5      .1       0  4156.2     .16       0
  4535.3      .1       0  4889.2     .16       0  4971.7     .05       0
  4994.2    .035       0  5000.2     .05       0  5080.8      .1       0
  5087.4     .16       0  5186.4     .05       0  5285.1      .1       0
  5383.8     .05       0  5482.6      .1       0  5662.4     .16       0
  5976.2      .1       0
Bank Sta=4994.2,5000.2
XS Rating Curve= 0 ,0
Exp/Cntr=0.3,0.1

Type RM Length L Ch R = 1 ,8769    ,624,624,624
BEGIN DESCRIPTION:
CALOHAN CREEK 19.0
END DESCRIPTION:
XS GIS Cut Line= 4
      2959465.96     10059019.17      2959955.56     10059638.99
      2960627.44     10059675.45      2961523.29     10060284.84
#Sta/Elev= 30
  3912.2 1133.53  4099.3 1115.61    4245 1103.98    4291 1094.38  4373.2 1086.68
  4408.5 1074.89  4429.3 1071.03  4536.7 1059.88    4562 1054.42  4607.4 1045.25
  4672.3 1032.97  4732.9 1027.65  4875.2 1020.82  4925.3 1009.46  5002.4 1008.55
  5005.2 1008.05  5008.4 1008.55  5034.6 1012.23  5158.8 1022.88  5265.8 1031.57
  5396.4 1055.95  5510.2 1067.19  5561.1 1081.34  5596.2 1083.93  5683.8 1089.86
  5730.5 1097.26  5935.2 1103.24  6249.9 1104.69  6354.2 1111.92  6458.4 1131.43
#Mann= 14 ,-1 , 0
  3912.2      .1       0  4099.3     .16       0    4291      .1       0
    4562     .16       0  4607.4      .1       0  4672.3     .16       0
  4732.9      .1       0  5002.4     .07       0  5008.4      .1       0
  5034.6     .05       0  5158.8      .1       0  5596.2     .16       0
  5730.5      .1       0  6249.9     .16       0
Bank Sta=5002.4,5008.4
XS Rating Curve= 0 ,0
Exp/Cntr=0.3,0.1

Type RM Length L Ch R = 1 ,8145    ,432,432,432
BEGIN DESCRIPTION:
CALOHAN CREEK 17.0
END DESCRIPTION:
XS GIS Cut Line= 4
      2958965.99     10059873.37      2959705.56      10060206.7
      2960653.48      10060331.7      2961334.64     10060560.49
#Sta/Elev= 30
  3700.8 1114.94  3732.8 1113.68  3884.4 1106.82  3930.6 1098.17  4110.9 1086.21
  4155.3 1075.42  4339.7 1062.93  4405.3  1055.6  4675.9 1030.67  4716.7 1023.25
  4769.7 1018.32  4874.6  1012.5  4959.9 1008.17  4996.1 1002.88  4998.9 1002.38
  5002.1 1002.88  5063.8  1007.7    5079 1015.19    5146 1019.75  5270.3  1029.6
  5311.8 1038.83  5368.1 1065.33  5402.6 1074.56  5422.7 1083.89    5484 1092.95
  5521.3 1104.95  5564.7 1107.74  5706.5 1120.73    5811 1137.64  6186.7  1152.3
#Mann= 14 ,-1 , 0
  3700.8      .1       0  3732.8     .16       0  4110.9      .1       0
  4405.3     .16       0  4769.7      .1       0  4874.6     .16       0
  4959.9      .1       0  4996.1     .07       0  5002.1      .1       0
    5079     .16       0    5146      .1       0  5270.3     .16       0
  5564.7      .1       0  5706.5     .16       0
Bank Sta=4996.1,5002.1
XS Rating Curve= 0 ,0
Exp/Cntr=0.3,0.1

Type RM Length L Ch R = 1 ,7713    ,440,440,440
BEGIN DESCRIPTION:
CALOHAN CREEK 16.0
END DESCRIPTION:
XS GIS Cut Line= 3
      2958913.92     10060040.05      2959742.02     10060612.95
      2961319.41     10060888.86
#Sta/Elev= 30
  3619.9 1116.27  3797.6 1106.67  3827.3 1099.92  3863.1 1096.98  4042.2 1088.73
  4077.5 1081.31  4122.6 1072.42  4229.5 1065.92  4358.5 1053.84  4480.8 1037.21
  4531.5 1026.92  4651.3 1022.17  4887.2 1015.64  4936.9 1010.83  4958.3 1004.03
  4995.9   999.4  4998.6   998.9  5001.9   999.4  5184.7 1018.34  5239.1 1044.12
  5298.6 1061.98  5358.1 1070.67  5394.8 1084.29  5445.6 1090.51  5496.3 1104.66
  5590.9  1117.1  5645.3  1131.1  5704.8  1140.9  5851.6 1154.59  6228.2  1159.6
#Mann= 7 ,-1 , 0
  3619.9     .16       0  4077.5      .1       0  4229.5     .16       0
  4651.3      .1       0  4936.9     .16       0  4995.9     .07       0
  5001.9     .16       0
Bank Sta=4995.9,5001.9
XS Rating Curve= 0 ,0
Exp/Cntr=0.3,0.1
