--- FLAT CREEK.prj (project) ---

Proj Title=FLAT CREEK Base Level Engineering
Current Plan=p01
Default Exp/Contr=0.3,0.1
English Units
Geom File=g01
Flow File=f01
Plan File=p01
Y Axis Title=Elevation
X Axis Title(PF)=Main Channel Distance
X Axis Title(XS)=Station
BEGIN DESCRIPTION:
FLAT CREEK
END DESCRIPTION:
DSS File=dss
DSS Export Rating Curves= 0
DSS Export Rating Curve Sorted= 0
DSS Export Volume Flow Curves= 0
DXF OffsetX= 0
DXF OffsetY= 0
DXF ScaleX= 1
DXF ScaleY= 10

--- FLAT CREEK.p01 (plan) ---

Plan Title=Multiple Run
Program Version=4.10
Short Identifier=Multiple Run
Geom File=g01
Flow File=f01
Subcritical Flow
K Sum by GR= 0
Std Step Tol= 0.01
Critical Tol= 0.01
Num of Std Step Trials= 20
Max Error Tol= 0.3
Flow Tol Ratio= 0.001
Split Flow NTrial= 30
Split Flow Tol= 0.02
Split Flow Ratio= 0.02
Log Output Level= 0
Friction Slope Method= 1
Unsteady Friction Slope Method= 2
Unsteady Bridges Friction Slope Method= 1
Parabolic Critical Depth
Global Vel Dist= 1 , 1 , 1
Global Log Level= 0
CheckData=True
Encroach Param=-1 ,0,0, 0
BEGIN DESCRIPTION:
Multiple Run
END DESCRIPTION:
Computation Interval=1HOUR
Output Interval=1HOUR
Run HTab= 0
Run UNet= 0
Run PostProcess= 0
Run WQNet= 0
UNET Theta= 1
UNET Theta Warmup= 1
UNET ZTol= 0.02
UNET ZSATol= 0.05
UNET MxIter= 20
UNET MaxInSteps= 0
UNET DtIC= 0
UNET DtMin= 0
UNET MaxCRTS= 20
UNET WFStab= 2
UNET SFStab= 1
UNET WFX= 1
UNET SFX= 1
UNET DSS MLevel= 4
UNET DZMax Abort= 100
UNET Convert EG Bridges= 0
UNET Use Existing IB Tables=-1
UNET Froude Reduction=False
UNET Froude Limit= 1
UNET Froude Power= 10
UNET Time Slicing=0,0, 5
UNET Junction Losses=0
Instantaneous Interval=1HOUR
DSS File=dss
Write IC File= 0
Write IC File at Sim End=0
Echo Input=False
Echo Parameters=False
Echo Output=False
Write Detailed= 0
WQ AD Non Conservative
WQ ULTIMATE=-1
WQ Max Comp Step=1HOUR
WQ Output Interval=15MIN
WQ Output Selected Increments= 0
WQ Output face flow=0
WQ Output face velocity=0
WQ Output face area=0
WQ Output face dispersion=0
WQ Output cell volume=0
WQ Output cell surface area=0
WQ Output cell continuity=0
WQ Output cumulative cell continuity=0
WQ Output face conc=0
WQ Output face dconc_dx=0
WQ Output face courant=0
WQ Output face peclet=0
WQ Output face adv mass=0
WQ Output face disp mass=0
WQ Output cell mass=0
WQ Output cell source sink temp=0
WQ Output cell source sink nsm=0
WQ Output MaxMinRange=-1
WQ Daily Max Min Mean=-1
WQ Daily Range=0
WQ Daily Time=0
WQ Create Restart=0
WQ Fixed Restart=0
WQ System Summary=0
WQ Use Fixed Temperature=0
Sorting and Armoring Iterations= 10
XS Update Threshold= 0.02
Hydraulics Update Threshold= 0.02
Energy Slope Method= 1
Volume Change Method= 0
XS Weighting Method= 0
Number of US Weighted Cross Sections= 1
Number of DS Weighted Cross Sections= 1
Upstream XS Weight=0.25
Main XS Weight=0.5
Downstream XS Weight=0.25
Number of DS XS's Weighted with US Boundary= 1
Upstream Boundary Weight= 1
Weight of XSs Associated with US Boundary= 0
Number of US XS's Weighted with DS Boundary= 1
Downstream Boundary Weight= 0.5
Weight of XSs Associated with DS Boundary= 0.5
Sediment Output Level= 4
Mass or Volume Output= 0
Output Increment Type= 1
Profile and TS Output Increment= 10
XS Output Flag= 0
XS Output Increment= 10
Disregard all LS=0
Disregard all Conn=0
Disregard all Breaches=0
Disregard all Pumps=0

--- FLAT CREEK.f01 (steady flow) ---

Flow Title=Multiple
Program Version=4.10
Number of Profiles= 7
Profile Names=10-year,25-year,50-year,1pct_min,100-year,1pct_plu,500-year
River Rch & RM=FLAT CREEK,Reach-1         ,70181
     935    1362    1736    1621    2192    2965    3507
River Rch & RM=FLAT CREEK,Reach-1         ,67581
    1398    2075    2677    2527    3417    4621    5586
River Rch & RM=FLAT CREEK,Reach-1         ,63117
    2015    3045    3975    3792    5128    6935    8569
River Rch & RM=FLAT CREEK,Reach-1         ,60639
    2317    3504    4577    4363    5900    7979    9845
River Rch & RM=FLAT CREEK,Reach-1         ,51781
    3129    4784    6294    6036    8164   11040   13793
River Rch & RM=FLAT CREEK,Reach-1         ,44472
    3387    5190    6838    6566    8879   12008   15037
River Rch & RM=FLAT CREEK,Reach-1         ,40393
    3565    5462    7195    6905    9339   12630   15801
River Rch & RM=FLAT CREEK,Reach-1         ,33871
    3845    5909    7799    7498   10141   13714   17220
River Rch & RM=FLAT CREEK,Reach-1         ,33435
    3845    5909    7799    7498   10141   13714   17220
River Rch & RM=FLAT CREEK,Reach-1         ,31798
    5600    8712   11595   11230   15187   20538   26165
River Rch & RM=FLAT CREEK,Reach-1         ,23653
    5874    9149   12187   11812   15974   21603   27559
River Rch & RM=FLAT CREEK,Reach-1         ,20999
    8159   12826   17195   16761   22667   30654   39547
River Rch & RM=FLAT CREEK,Reach-1         ,15583
    8217   12906   17292   16844   22779   30807   39689
River Rch & RM=FLAT CREEK,Reach-1         ,10584
    8238   12923   17300   16837   22769   30793   39597
River Rch & RM=FLAT CREEK,Reach-1         ,5147
    8877   13950   18697   18215   24633   33314   42924
River Rch & RM=FLAT CREEK,Reach-1         ,4817
    8877   13950   18697   18215   24633   33314   42924
Boundary for River Rch & Prof#=FLAT CREEK,Reach-1         , 1
Up Type= 0
Dn Type= 3
Dn Slope=0.005
Boundary for River Rch & Prof#=FLAT CREEK,Reach-1         , 2
Up Type= 0
Dn Type= 3
Dn Slope=0.005
Boundary for River Rch & Prof#=FLAT CREEK,Reach-1         , 3
Up Type= 0
Dn Type= 3
Dn Slope=0.005
Boundary for River Rch & Prof#=FLAT CREEK,Reach-1         , 4
Up Type= 0
Dn Type= 3
Dn Slope=0.005
Boundary for River Rch & Prof#=FLAT CREEK,Reach-1         , 5
Up Type= 0
Dn Type= 3
Dn Slope=0.005
Boundary for River Rch & Prof#=FLAT CREEK,Reach-1         , 6
Up Type= 0
Dn Type= 3
Dn Slope=0.005
Boundary for River Rch & Prof#=FLAT CREEK,Reach-1         , 7
Up Type= 0
Dn Type= 3
Dn Slope=0.005
DSS Import GetInterval= 0
DSS Import GetPeak= 0
DSS Import FillOption= 0

--- FLAT CREEK.g01 (geometry) ---

Geom Title=Existing Conditions
Program Version=4.10

River Reach=FLAT CREEK      ,Reach-1
Reach XY= 30
      2955358.07     10041054.21      2954841.33     10044052.42
      2957398.47     10046593.73      2957744.57       10050033.
       2956307.9     10052403.58      2955182.52     10052997.72
      2955016.51     10054222.79      2954137.83     10054432.12
      2954815.43     10055656.87      2954420.06     10057488.07
       2955086.4     10057694.01      2955518.33     10059419.04
      2954843.55     10064512.09      2956366.08      10066618.1
      2960280.85     10067179.67      2961283.91     10068611.91
      2962994.81     10067701.64      2963542.82     10069480.01
      2965837.05     10067873.48      2968230.09     10069562.25
      2968487.41     10070893.42      2967320.21     10071450.68
      2967147.71     10072326.74      2968732.51     10072184.48
      2969111.92     10073010.37      2966992.96     10075646.91
      2966291.41      10078734.7      2966848.98     10079717.66
      2965448.87     10082173.16      2966608.09      10083466.9

Type RM Length L Ch R = 1 ,70181   ,783,783,783
BEGIN DESCRIPTION:
FLAT CREEK 143.0
END DESCRIPTION:
XS GIS Cut Line= 4
       2954595.5     10041111.56      2955179.25     10041150.62
      2955665.36     10041152.79      2956299.08     10041063.81
#Sta/Elev= 30
  4225.5 1319.43  4298.6 1312.42    4459 1304.58  4589.3 1294.34  4637.5 1294.16
  4693.5  1295.2  4778.5 1296.34  4812.7 1293.55  4839.8 1288.93  4939.8 1281.73
  4978.9 1274.09 4984.43 1269.01  4989.8 1265.65  4996.8  1264.4  4999.5  1263.9
  5002.8  1264.4 5013.07 1268.76  5019.8 1272.68  5029.8 1274.59    5067 1277.12
  5149.8 1283.38  5219.8 1301.39  5269.8 1307.86  5350.3 1313.62  5370.5 1318.22
  5401.8  1320.9  5431.1 1326.45    5522 1333.24  5879.7 1346.46  5936.6 1349.43
#Mann= 8 ,-1 , 0
  4225.5     .05       0  4637.5     .16       0  4693.5     .05       0
  4978.9     .16       0  4996.8     .07       0  5002.8     .16       0
    5067      .1       0  5879.7     .16       0
Bank Sta=4984.43,5013.07
XS Rating Curve= 0 ,0
Exp/Cntr=0.3,0.1

Type RM Length L Ch R = 1 ,69398   ,105,105,105
BEGIN DESCRIPTION:
Mapping XS 1582488d
END DESCRIPTION:
XS GIS Cut Line= 4
      2954442.23     10041577.63      2955191.36     10041778.83
      2955561.65     10041778.83      2956167.43     10041549.79
#Sta/Elev= 30
  4088.9 1317.89  4211.6 1314.63  4326.4 1309.58  4374.9 1305.48  4675.9 1295.21
  4830.7 1283.75  4871.7  1277.5  4951.7 1268.67  4961.7  1264.3  4971.7 1261.85
  4980.6 1258.79  4991.7 1252.31  4998.7 1249.92  5001.4 1249.42  5004.7 1249.92
  5051.7 1261.87  5081.7 1270.72  5111.7    1275  5151.7 1289.59  5171.7 1293.33
  5195.3 1295.77  5230.8 1298.69  5321.1    1302    5456 1311.78  5491.5 1316.28
  5546.5 1319.12  5584.3 1323.09  5741.7 1329.69  5777.2    1333  5882.5 1334.66
#Mann= 5 ,-1 , 0
  4088.9      .1       0  4980.6     .16       0  4998.7     .07       0
  5004.7     .16       0  5195.3      .1       0
Bank Sta=4971.7,5051.7
XS Rating Curve= 0 ,0
Exp/Cntr=0.3,0.1

Type RM Length L Ch R = 1 ,69293   ,72,72,72
BEGIN DESCRIPTION:
Mapping XS efe637bd
END DESCRIPTION:
XS GIS Cut Line= 4
      2954404.56     10041641.08       2955233.5     10041875.45
      2955476.56     10041868.94      2956163.97     10041632.57
#Sta/Elev= 30
  4072.1 1322.94  4140.3  1321.1  4208.3 1316.68  4359.7 1311.09  4393.7 1307.36
  4466.8 1303.82  4678.9 1296.45  4720.2 1291.44  4823.6  1284.3  4910.7 1273.73
  4968.5 1262.99  4995.5 1260.82  4998.3 1260.32  5001.5 1260.82  5020.8 1261.31
  5038.5 1263.03  5108.6 1261.23  5118.6 1267.92  5128.6 1281.12  5138.6 1288.31
  5158.6 1292.79  5221.4 1297.95  5316.2 1300.46  5379.6 1304.92  5538.2  1312.5
  5581.5 1318.35  5695.8  1321.6  5739.2 1325.51  5844.9 1328.92  5903.6 1332.86
#Mann= 7 ,-1 , 0
  4072.1      .1       0  4823.6     .16       0  4910.7      .1       0
  4995.5     .07       0  5001.5      .1       0  5020.8     .16       0
  5221.4      .1       0
#XS Ineff= 2 , 0
                         5046.59          1263.3
Permanent Ineff=
       T       T
Bank Sta=4968.5,5038.5
XS Rating Curve= 0 ,0
Exp/Cntr=0.3,0.1

Type RM Length L Ch R = 1 ,69221   ,126,126,126
BEGIN DESCRIPTION:
FLAT CREEK 142.0
END DESCRIPTION:
XS GIS Cut Line= 4
       2954371.6     10041678.23      2955234.17     10041939.36
      2955527.41     10041928.66      2956193.11     10041706.04
#Sta/Elev= 30
  4010.1 1326.23    4187 1320.64  4214.7 1317.28    4291 1314.37  4389.8 1307.13
  4654.6 1294.82  4748.6 1286.65  4805.9 1283.88  4890.6 1271.39  4909.9 1265.42
  4935.6  1261.9  4955.7 1255.79 4980.68 1252.02  4995.7 1246.77  5012.7 1246.19
  5015.4 1245.69  5018.7 1246.19  5025.7 1246.51 5039.77 1251.89  5055.7 1258.23
  5095.7 1284.45  5135.8 1292.04  5204.1 1296.59  5311.3  1299.5  5365.7 1303.56
  5574.9 1311.02  5618.4 1314.73  5739.5 1319.51  5807.9 1325.62  5906.7 1328.29
#Mann= 5 ,-1 , 0
  4010.1      .1       0  4890.6     .16       0  5012.7     .07       0
  5018.7     .16       0  5204.1      .1       0
Bank Sta=4980.68,5039.77
XS Rating Curve= 0 ,0
Exp/Cntr=0.3,0.1

Type RM Length L Ch R = 1 ,69095   ,373,373,373
BEGIN DESCRIPTION:
FLAT CREEK 141.0
END DESCRIPTION:
XS GIS Cut Line= 4
      2954420.53     10041833.78       2955042.1     10041903.22
      2955385.85     10042125.45      2956229.63     10042087.25
#Sta/Elev= 30
    4118 1329.39  4257.3 1323.32  4317.2 1316.13    4458 1306.48  4679.4 1295.13
  4770.4  1287.2    4849 1283.12  4927.9 1272.32  4957.8 1265.28    4973 1250.94
  4991.1 1242.93  4993.8 1242.43  4997.1 1242.93  5024.4 1244.63  5030.4 1245.73
  5036.8 1249.31  5051.5 1253.24  5066.6 1261.54  5072.6 1262.56  5145.2 1266.79
  5175.4 1273.37  5269.5  1285.2  5345.6 1287.31  5415.6 1284.94  5445.7 1286.33
  5475.7 1291.45  5521.5 1296.08  5625.9 1299.96  5665.9 1303.67  5997.4 1323.34
#Mann= 5 ,-1 , 0
    4118      .1       0  4927.9     .16       0  4991.1     .07       0
  4997.1     .16       0  5269.5      .1       0
Bank Sta=4973,5036.8
XS Rating Curve= 0 ,0
Exp/Cntr=0.3,0.1

Type RM Length L Ch R = 1 ,68722   ,348,348,348
BEGIN DESCRIPTION:
FLAT CREEK 140.0
END DESCRIPTION:
XS GIS Cut Line= 3
      2954507.38     10042337.25      2955000.43     10042396.28
      2956101.16     10042396.28
#Sta/Elev= 30
  4334.4 1317.06  4360.5 1314.58  4395.9 1310.28  4436.2 1300.87  4496.6 1295.39
  4587.3 1295.03  4627.6 1292.93  4758.5 1293.24  4788.7 1288.79  4818.9 1289.18
  4862.7 1285.92    4889 1284.34    4909  1279.6    4939 1254.56    4959 1244.38
    4996 1237.55  4998.8 1237.05    5002 1237.55    5009 1239.03    5019 1245.16
    5029 1252.15    5039 1255.53  5180.2 1263.74    5209 1265.93    5239 1271.68
    5409  1283.6    5479 1291.31    5799 1310.26    5889 1319.04  5931.7 1321.15
#Mann= 6 ,-1 , 0
  4334.4     .16       0  4360.5      .1       0  4862.7     .16       0
    4996     .07       0    5002     .16       0  5180.2      .1       0
Bank Sta=4959,5019
XS Rating Curve= 0 ,0
Exp/Cntr=0.3,0.1

Type RM Length L Ch R = 1 ,68374   ,341,341,341
BEGIN DESCRIPTION:
FLAT CREEK 139.0
END DESCRIPTION:
XS GIS Cut Line= 4
      2954486.55     10042410.17      2954826.82     10042496.97
       2955128.9     10042694.89      2956057.89     10042708.76
#Sta/Elev= 30
  4110.2 1310.32  4141.4  1308.4  4174.1 1299.56  4231.4 1294.92  4411.5 1292.81
  4452.7 1295.42  4459.6 1293.95  4466.9 1296.93    4482  1293.2  4524.2 1293.26
  4554.4 1288.66  4596.6 1288.21  4682.2 1280.17  4832.1 1257.75  4872.1 1248.76
  4892.1 1241.09  4922.1 1237.77  4989.1  1231.4  4991.8  1230.9  4995.1  1231.4
  5012.1 1232.73  5022.1 1238.05  5032.1 1247.78  5042.1 1251.98  5112.1 1261.81
  5212.1 1282.61  5292.1 1292.39  5430.4 1298.19  5502.1 1305.28  5751.6 1317.93
#Mann= 6 ,-1 , 0
  4110.2     .16       0  4231.4      .1       0  4682.2     .16       0
  4989.1     .07       0  4995.1     .16       0  5430.4      .1       0
Bank Sta=4922.1,5022.1
XS Rating Curve= 0 ,0
Exp/Cntr=0.3,0.1

Type RM Length L Ch R = 1 ,68033   ,452,452,452
BEGIN DESCRIPTION:
FLAT CREEK 138.0
END DESCRIPTION:
XS GIS Cut Line= 4
      2954684.44     10042943.15      2955087.24     10042955.31
       2955503.9     10043125.45      2955933.95     10043063.02
#Sta/Elev= 30
  4414.3 1291.57  4448.3 1292.11  4468.4 1287.55  4498.4 1288.52  4528.4 1282.53
  4558.4 1281.62  4608.4 1273.32  4673.7 1257.04  4688.5 1253.24  4698.5 1245.85
  4710.3 1245.25  4748.5 1244.58  4788.5 1249.75  4872.6 1252.13  4902.7 1248.92
  4937.5 1237.98  4961.5  1234.2  4999.2  1225.1    5002  1224.6  5005.2  1225.1
  5033.6 1233.97    5039 1236.04  5045.4 1242.83  5056.2 1257.52    5063 1270.08
  5068.4 1271.91  5172.1 1276.62    5218 1280.93  5433.6 1289.97  5701.9 1294.97
#Mann= 6 ,-1 , 0
  4414.3     .16       0  4673.7      .1       0  4710.3     .16       0
  4999.2     .07       0  5005.2     .16       0  5172.1      .1       0
#XS Ineff= 2 , 0
          4871.7 1252.24
Permanent Ineff=
       T       T
Bank Sta=4961.5,5033.6
XS Rating Curve= 0 ,0
Exp/Cntr=0.3,0.1

Type RM Length L Ch R = 1 ,67581   ,688,688,688
BEGIN DESCRIPTION:
FLAT CREEK 137.0
END DESCRIPTION:
XS GIS Cut Line= 4
      2954371.93     10042927.51      2955017.79     10043338.99
      2955189.67     10043521.28      2955735.02     10043692.68
#Sta/Elev= 30
  4331.3 1302.51  4354.5 1300.58  4362.8 1291.11    4385  1287.9  4694.8 1287.12
  4739.6 1282.01  4797.2 1282.16  4875.9 1276.64    4920 1272.91  4933.5 1262.57
  4936.4 1257.57  4942.8 1246.53  4955.6 1230.97  4963.9 1226.68  4979.2 1221.53
  4997.3 1220.29  5000.1 1219.79  5003.3 1220.29  5020.7 1225.22  5027.4 1227.43
  5122.1 1233.85  5178.7 1243.89  5291.8 1246.42  5410.2 1249.56  5482.7 1267.05
  5506.7 1270.43    5598 1273.87  5692.3 1281.85  5854.9 1290.53  5919.3 1293.39
#Mann= 8 ,-1 , 0
  4331.3      .1       0  4936.4     .16       0  4997.3     .07       0
  5003.3     .16       0  5020.7      .1       0  5291.8     .16       0
  5506.7      .1       0  5854.9     .16       0
Bank Sta=4963.9,5027.4
XS Rating Curve= 0 ,0
Exp/Cntr=0.3,0.1

Type RM Length L Ch R = 1 ,66893   ,450,450,450
BEGIN DESCRIPTION:
FLAT CREEK 136.0
END DESCRIPTION:
XS GIS Cut Line= 3
      2954715.72     10043474.43      2954996.96     10044010.86
       2955584.5     10043969.27
#Sta/Elev= 30
  4518.5 1272.74  4601.1 1272.83  4623.2 1270.69  4661.6 1260.87  4667.3 1260.66
  4683.7 1254.42  4705.7 1248.82  4749.9 1241.18  4755.5 1238.84  4771.9 1237.78
  4788.3 1233.61    4800 1228.31  4822.6  1224.2  4970.5 1217.97  4986.9 1213.52
    5003 1211.43  5003.5 1211.43 5018.86 1218.31  5025.3 1221.46  5037.1 1222.31
    5226 1217.62  5293.5 1216.79  5326.2 1218.24  5346.3 1223.76  5386.4 1244.42
  5416.4 1265.69  5426.5  1271.1    5509 1275.31  5566.8 1280.66  5713.2 1285.74
#Mann= 5 ,-1 , 0
  4518.5      .1       0  4970.5     .05       0  4970.5     .07       0
  5003.5     .16       0    5509      .1       0
#XS Ineff= 2 , 0
                         5037.95         1222.32
Permanent Ineff=
       T       T
Bank Sta=4970.5,5018.86
XS Rating Curve= 0 ,0
Exp/Cntr=0.3,0.1

Type RM Length L Ch R = 1 ,66443   ,772,772,772
BEGIN DESCRIPTION:
FLAT CREEK 135.0
END DESCRIPTION:
XS GIS Cut Line= 4
      2954470.92     10044635.86      2954825.08     10044338.99
      2955179.25     10044135.86      2955637.54     10044016.08
#Sta/Elev= 30
  4384.3 1283.52  4426.6 1278.53  4440.9 1274.58    4519 1259.56  4581.4  1251.5
  4596.3 1248.21  4693.5 1243.47    4774 1241.15  4824.7 1235.53  4849.8 1235.29
  4947.9 1233.94  4963.7 1230.29  4985.3 1213.81  4997.2 1207.44  4999.9 1206.94
  5003.2 1207.44  5028.4 1214.18    5109 1216.44  5232.2 1214.69  5295.2 1217.11
  5315.9 1222.06  5321.8 1228.06  5326.9 1227.43    5357  1248.2  5362.2 1245.27
  5367.6 1259.56  5377.9 1272.91  5482.7 1280.85  5646.7 1285.22  5728.4  1290.8
#Mann= 10 ,-1 , 0
  4384.3     .16       0  4440.9      .1       0  4581.4     .16       0
  4596.3      .1       0  4693.5     .05       0  4849.8      .1       0
  4997.2     .07       0  5003.2      .1       0  5232.2     .16       0
  5482.7      .1       0
#XS Ineff= 2 , 0
                         5108.18         1216.65
Permanent Ineff=
       T       T
Bank Sta=4985.3,5028.4
XS Rating Curve= 0 ,0
Exp/Cntr=0.3,0.1

Type RM Length L Ch R = 1 ,65671   ,577,577,577
BEGIN DESCRIPTION:
FLAT CREEK 133.0
END DESCRIPTION:
XS GIS Cut Line= 4
      2954554.28     10044854.61        2955148.     10044828.57
      2955293.83     10044578.57      2955746.96      10044161.9
#Sta/Elev= 30
  4283.9 1284.08  4318.1 1281.84  4348.1 1278.08  4358.2    1274  4430.8 1265.87
  4508.3 1251.36  4563.5 1245.41  4625.1 1240.17  4738.5 1233.26  4910.8 1230.08
  4941.7 1226.48  4958.7 1221.18  4969.5 1217.83  4976.4 1211.55    4991 1201.27
  4996.6 1201.11  4999.3 1200.61  5002.6 1201.11  5012.5 1205.53  5071.2 1212.25
  5195.6 1214.58  5323.2 1228.11    5351 1233.96  5415.1 1267.73  5436.1 1273.43
    5507 1274.26  5601.1  1282.9  5662.9 1285.37  5698.1 1290.25  5783.2 1292.17
#Mann= 8 ,-1 , 0
  4283.9      .1       0  4430.8     .16       0  4563.5      .1       0
  4625.1     .05       0  4958.7     .16       0  4996.6     .07       0
  5002.6     .16       0  5601.1      .1       0
Bank Sta=4976.4,5071.2
XS Rating Curve= 0 ,0
Exp/Cntr=0.3,0.1

Type RM Length L Ch R = 1 ,65094   ,506,506,506
BEGIN DESCRIPTION:
FLAT CREEK 132.0
END DESCRIPTION:
XS GIS Cut Line= 3
      2954580.25     10044917.11      2955726.12      10044906.7
      2956080.32     10044479.57
#Sta/Elev= 30
  3982.2 1283.71  4020.4 1279.78  4030.4 1275.45  4065.7 1273.57  4100.1 1269.68
  4170.4 1261.98  4297.5 1242.87  4450.4 1234.11  4668.2 1226.69  4801.5 1219.57
  4904.8 1217.03  4950.5 1207.02  4997.5 1196.94  5000.2 1196.44  5003.5 1196.94
  5010.5 1198.05  5020.5 1204.01  5030.5 1211.52  5040.5 1215.19  5090.5 1222.95
  5120.5 1229.13  5126.8 1232.23  5133.3 1232.23  5167.7 1250.73  5202.9 1273.45
  5223.7 1284.49    5238 1289.24  5266.7  1292.9  5386.3 1294.03    5683 1302.14
#Mann= 9 ,-1 , 0
  3982.2     .16       0  4065.7      .1       0  4100.1     .16       0
  4297.5     .05       0  4668.2      .1       0  4801.5     .16       0
  4997.5     .07       0  5003.5     .16       0  5386.3      .1       0
Bank Sta=4950.5,5020.5
XS Rating Curve= 0 ,0
Exp/Cntr=0.3,0.1

Type RM Length L Ch R = 1 ,64588   ,206,206,206
BEGIN DESCRIPTION:
FLAT CREEK 131.0
END DESCRIPTION:
XS GIS Cut Line= 4
      2955064.68     10045828.56      2955799.04     10045302.53
      2956033.42      10044969.2      2956236.55     10044411.88
#Sta/Elev= 30
  3903.1 1275.73  3997.3 1268.61  4053.3 1266.14  4145.4  1255.8  4210.5 1252.47
  4231.4 1247.92  4311.2 1245.15  4324.9 1241.56  4346.9 1237.04  4447.6 1229.94
  4837.1 1216.72    4879 1216.38  4934.6 1210.31  4963.9 1203.14  4976.4  1196.1
  4996.9 1191.88  4999.7 1191.38  5002.9 1191.88  5012.8 1193.19  5026.9 1200.63
  5056.5 1222.01  5077.5 1225.21  5098.4 1236.11  5107.1 1242.59  5121.9 1258.61
    5128 1274.71  5142.8 1286.92  5163.7 1290.02  5293.6 1293.31  5807.1 1307.15
#Mann= 8 ,-1 , 0
  3903.1     .16       0  3997.3      .1       0  4324.9     .05       0
  4837.1      .1       0    4879     .16       0  4996.9     .07       0
  5002.9     .16       0  5293.6      .1       0
Bank Sta=4963.9,5026.9
XS Rating Curve= 0 ,0
Exp/Cntr=0.3,0.1

Type RM Length L Ch R = 1 ,64382   ,430,430,430
BEGIN DESCRIPTION:
FLAT CREEK 130.0
END DESCRIPTION:
XS GIS Cut Line= 3
      2955184.47     10045922.31      2956007.37      10045406.7
      2956460.51     10044469.16
#Sta/Elev= 30
  3870.4 1274.64  4094.8 1254.74  4134.7 1252.86  4177.3 1246.12    4235 1245.03
  4271.5  1235.9  4365.8  1229.1  4572.2 1221.11  4643.3 1218.84  4764.5 1215.86
  4898.1 1212.19  4943.3 1207.36  4971.5 1199.92  4978.1 1195.06  4997.3 1189.89
    5000 1189.39  5003.3 1189.89  5016.7  1191.7  5033.6 1201.41  5044.8 1210.12
    5078 1219.99  5100.2 1230.64  5152.2 1261.95  5189.1 1278.61  5211.3 1281.38
  5294.6 1281.17  5408.7 1288.35  5441.5 1288.17    5779 1293.65  5882.8 1300.87
#Mann= 10 ,-1 , 0
  3870.4      .1       0  4094.8     .05       0  4572.2      .1       0
  4643.3     .05       0  4764.5     .16       0  4997.3     .07       0
  5003.3     .16       0  5294.6      .1       0  5408.7     .16       0
  5441.5      .1       0
Bank Sta=4971.5,5033.6
XS Rating Curve= 0 ,0
Exp/Cntr=0.3,0.1

Type RM Length L Ch R = 1 ,63952   ,457,457,457
BEGIN DESCRIPTION:
FLAT CREEK 129.0
END DESCRIPTION:
XS GIS Cut Line= 4
      2955189.67     10046068.15      2956028.21     10045588.99
      2956642.79     10045547.32      2956912.62     10045287.87
#Sta/Elev= 30
  3712.7 1283.64  3780.4 1275.56  3856.5 1269.25  3934.6 1262.64  3977.8 1260.77
  3999.4 1256.93  4068.4 1251.63  4079.9 1248.58  4154.8 1243.88  4176.4 1237.74
  4206.6 1232.11  4546.2 1218.11    4750 1212.37  4959.4 1197.33  4976.2 1190.56
  4996.5 1187.18  4999.2 1186.68  5002.5 1187.18 5017.05 1196.97  5019.5 1201.01
  5029.5 1203.35  5099.7 1208.29  5139.8 1215.58  5189.9 1236.12    5240 1262.09
  5280.1 1279.91  5330.9 1285.02  5371.7 1287.78  5583.9 1292.56  5668.8 1299.07
#Mann= 8 ,-1 , 0
  3712.7     .16       0  3856.5      .1       0  4079.9     .05       0
  4546.2      .1       0    4750     .16       0  4996.5     .07       0
  5002.5     .16       0  5330.9      .1       0
Bank Sta=4959.4,5017.05
XS Rating Curve= 0 ,0
Exp/Cntr=0.3,0.1

Type RM Length L Ch R = 1 ,63495   ,378,378,378
BEGIN DESCRIPTION:
FLAT CREEK 128.0
END DESCRIPTION:
XS GIS Cut Line= 3
      2955564.68     10046354.61      2956533.42      10046031.7
      2956788.62     10045609.82
#Sta/Elev= 30
  3798.3 1264.19  3894.3 1259.27  3941.3 1255.99  4020.7 1248.73  4044.7  1244.9
  4096.8 1242.14  4139.6 1234.04  4177.8 1230.79  4283.3 1221.54  4465.4 1213.52
  4836.7  1206.7  4852.1 1204.82  4869.3 1199.97  4953.1 1196.69  4968.6 1192.98
  4980.7 1185.44  4992.8 1182.77  4995.6 1182.27  4998.8 1182.77  5017.2 1185.01
  5032.7  1189.7 5035.91 1192.32  5048.2 1203.97    5054 1207.02    5085 1216.97
  5106.4 1225.97  5170.4 1257.48  5214.4 1276.51    5250 1284.77  5312.5 1287.51
#Mann= 10 ,-1 , 0
  3798.3      .1       0  3894.3     .16       0  3941.3      .1       0
  4020.7     .16       0  4177.8      .1       0  4283.3     .05       0
  4465.4      .1       0  4869.3     .16       0  4992.8     .07       0
  4998.8     .16       0
Bank Sta=4968.6,5035.91
XS Rating Curve= 0 ,0
Exp/Cntr=0.3,0.1

Type RM Length L Ch R = 1 ,63117   ,488,488,488
BEGIN DESCRIPTION:
FLAT CREEK 127.0
END DESCRIPTION:
XS GIS Cut Line= 3
      2955726.12     10046401.49      2956736.54     10046255.65
      2957111.57      10045984.8
#Sta/Elev= 30
  3791.6 1255.39  4001.9 1242.32  4035.4 1237.85  4156.8 1231.79  4186.9 1226.14
  4232.2 1218.38  4287.2 1215.93  4438.1 1211.01  4448.8 1210.56  4688.4 1206.68
  4828.8  1202.4  4858.3 1198.32  4908.2 1198.69    4938 1196.42  4958.8 1186.74
  4997.6 1179.06  5000.3 1178.56  5003.6 1179.06  5023.8 1187.69  5033.3 1190.96
  5065.6 1201.46  5080.3 1211.35  5115.9 1220.45  5136.8 1230.55  5166.2 1247.57
  5172.6 1256.91  5180.9 1263.64  5195.6  1270.3  5216.5 1277.11  5275.1 1279.74
#Mann= 12 ,-1 , 0
  3791.6      .1       0  4001.9     .16       0  4035.4      .1       0
  4186.9     .16       0  4287.2      .1       0  4438.1     .16       0
  4448.8      .1       0  4688.4     .05       0  4908.2      .1       0
  4997.6     .07       0  5003.6      .1       0  5033.3     .16       0
Bank Sta=4958.8,5023.8
XS Rating Curve= 0 ,0
Exp/Cntr=0.3,0.1

Type RM Length L Ch R = 1 ,62629   ,579,579,579
BEGIN DESCRIPTION:
FLAT CREEK 126.0
END DESCRIPTION:
XS GIS Cut Line= 4
      2956455.28     10047062.95      2957054.25     10046693.15
      2957184.46     10046427.53      2957262.57      10046073.4
#Sta/Elev= 30
    4159 1244.86  4225.8 1241.48  4241.2  1235.9  4268.5 1230.04  4314.5 1224.52
  4430.4 1217.51  4621.4  1209.5  4735.4 1203.24  4926.4 1196.51  4962.5  1192.2
  4971.4 1189.06 4980.91 1179.52  4984.8 1175.97  4990.9 1174.14  4993.7 1173.64
  4996.9 1174.14  5029.3 1179.04  5083.9 1186.78  5151.4 1192.48  5193.4 1198.03
  5248.3 1209.49  5254.8 1213.51  5285.5 1223.12  5299.2 1229.54    5347 1247.98
  5384.5 1257.89  5418.7 1264.27    5477 1270.98  5505.6 1272.53  5521.4 1273.47
#Mann= 6 ,-1 , 0
    4159     .05       0  4621.4      .1       0  4990.9     .07       0
  4996.9      .1       0  5299.2     .16       0  5505.6      .1       0
Bank Sta=4980.91,5029.3
XS Rating Curve= 0 ,0
Exp/Cntr=0.3,0.1

Type RM Length L Ch R = 1 ,62050   ,475,475,475
BEGIN DESCRIPTION:
FLAT CREEK 125.0
END DESCRIPTION:
XS GIS Cut Line= 4
      2956575.08     10047151.49        2957148.     10046875.45
      2957908.42     10046870.24      2958423.77     10046979.55
#Sta/Elev= 30
  4073.3 1244.22  4126.4 1241.26  4143.4 1236.41  4171.6 1223.52  4186.6 1222.08
  4206.2 1218.97  4432.8 1205.59    4522 1199.35  4697.4 1191.33  4849.7 1190.62
  4938.7 1176.88  4939.7 1176.54  4949.7 1172.68  4976.7 1169.91  4979.5 1169.41
  4982.7 1169.91  5019.7 1170.84  5037.4 1175.95  5059.7 1181.74  5079.7 1179.65
  5259.7 1190.71  5309.7 1197.15  5432.1 1202.41    5664 1219.96  5687.8 1218.72
  5706.7 1220.73  5725.3 1229.86  5800.9 1239.08  5868.4 1251.03  5996.5 1259.87
#Mann= 11 ,-1 , 0
  4073.3      .1       0  4186.6     .05       0  4206.2      .1       0
  4432.8     .05       0    4522      .1       0  4938.7     .05       0
  4976.7    .035       0  4982.7     .05       0  5037.4     .16       0
  5432.1     .05       0  5687.8      .1       0
Bank Sta=4939.7,5037.4
XS Rating Curve= 0 ,0
Exp/Cntr=0.3,0.1

Type RM Length L Ch R = 1 ,61575   ,486,486,486
BEGIN DESCRIPTION:
FLAT CREEK 124.0
END DESCRIPTION:
XS GIS Cut Line= 2
      2956804.29      10047344.2      2958382.38      10047349.4
#Sta/Elev= 30
  4385.7 1246.52  4409.9 1244.75  4459.9 1235.31  4499.9 1221.06  4559.9 1207.71
  4639.9 1196.86  4704.2 1192.04  4840.1 1183.26  4919.9 1179.74  4939.9 1176.34
  4949.9  1172.6  4969.9  1167.5  4996.9 1164.02  4999.6 1163.52  5002.9 1164.02
  5029.9 1167.87  5049.9 1174.29  5059.9 1177.42  5099.9 1180.56  5204.8 1183.78
  5234.7 1185.21  5333.4 1194.59    5432 1199.92  5612.9 1207.56  5669.9 1213.32
  5689.9 1217.23  5729.9 1217.31  5739.9 1220.18  5799.9 1226.17  5963.8 1254.23
#Mann= 10 ,-1 , 0
  4385.7     .05       0  4704.2      .1       0  4840.1     .16       0
  4996.9     .07       0  5002.9     .16       0  5204.8      .1       0
  5234.7     .16       0  5333.4      .1       0    5432     .05       0
  5612.9      .1       0
Bank Sta=4949.9,5049.9
XS Rating Curve= 0 ,0
Exp/Cntr=0.3,0.1

Type RM Length L Ch R = 1 ,61089   ,450,450,450
BEGIN DESCRIPTION:
FLAT CREEK 123.0
END DESCRIPTION:
XS GIS Cut Line= 4
      2956825.07     10047682.73      2957309.46     10047792.11
      2957580.29     10047885.86      2958413.57     10047771.29
#Sta/Elev= 30
  4406.2 1252.61  4429.8 1252.21  4482.7 1250.83  4553.2 1242.36  4569.1 1236.29
  4604.5 1228.74  4631.6 1217.89    4709  1191.8  4731.8 1187.88    4871 1174.61
  4909.2 1168.29  4944.1 1164.56  4975.8  1165.2  5004.6 1158.71  5007.3 1158.21
  5010.6 1158.71 5035.11 1168.84  5044.9 1172.53  5083.6 1173.88  5298.6 1179.13
  5500.2 1193.39  5713.5 1207.71  5742.7 1210.36    5773 1209.67  5793.2 1213.83
    5884 1220.14  5900.8  1224.4  5905.8 1222.17  5975.2 1232.56  6030.5  1245.1
#Mann= 11 ,-1 , 0
  4406.2      .1       0  4429.8     .16       0  4631.6      .1       0
  4731.8     .05       0  4909.2     .16       0  5004.6     .07       0
  5010.6     .16       0  5083.6      .1       0  5500.2     .05       0
  5713.5      .1       0  5975.2     .16       0
Bank Sta=4909.2,5035.11
XS Rating Curve= 0 ,0
Exp/Cntr=0.3,0.1

Type RM Length L Ch R = 1 ,60639   ,647,647,647
BEGIN DESCRIPTION:
FLAT CREEK 122.0
END DESCRIPTION:
XS GIS Cut Line= 4
      2956590.72      10048094.2      2957043.83     10048198.36
      2957705.29     10048276.49      2958632.38     10047995.24
#Sta/Elev= 30
  4366.5 1256.79  4405.2 1251.94  4466.8 1249.97  4511.7 1241.67  4538.6 1232.16
  4564.8 1218.76  4612.7 1207.14  4682.3 1203.46  4789.2 1193.69  4831.2 1179.85
  4936.8 1172.99  4977.1 1165.49  4994.2 1153.59    4997 1153.09  5000.2 1153.59
  5038.5 1160.75  5091.6  1161.1  5138.2 1164.66  5213.6  1170.4  5565.1 1178.12
  5793.4 1188.32  5973.2 1202.12    5992 1202.66  6012.9 1208.44    6111 1220.19
    6182 1240.18  6242.6 1242.93  6305.5 1250.18    6434 1253.94  6466.3 1252.59
#Mann= 9 ,-1 , 0
  4366.5      .1       0  4511.7     .05       0  4994.2    .035       0
  5000.2     .05       0  5038.5     .16       0  5213.6      .1       0
  5565.1     .05       0  5973.2      .1       0    6434     .16       0
Bank Sta=4977.1,5138.2
XS Rating Curve= 0 ,0
Exp/Cntr=0.3,0.1

Type RM Length L Ch R = 1 ,59992   ,343,343,343
BEGIN DESCRIPTION:
FLAT CREEK 121.0
END DESCRIPTION:
XS GIS Cut Line= 4
      2956549.08     10048599.41        2957273.     10048755.65
      2957746.96     10048755.65      2958517.81     10048557.73
#Sta/Elev= 30
  4103.9 1252.11  4192.9 1252.07  4348.8 1241.44  4398.5 1235.14    4429 1233.03
    4492 1212.25  4512.5 1210.92  4594.3 1195.79  4635.2 1180.38  4669.3 1173.39
  4839.6 1160.31  4959.1 1157.57    5007 1149.59  5009.7 1149.09    5013 1149.59
    5020 1150.81    5030 1159.77  5066.3 1165.49    5165 1167.11    5275 1171.25
  5364.2 1175.64  5498.4 1183.51  5631.3 1189.37  5753.8 1198.74  5794.9 1199.18
  5870.7 1206.37  5911.4 1214.52  5960.1 1231.16  6001.4 1240.19  6114.3 1246.92
#Mann= 12 ,-1 , 0
  4103.9      .1       0  4398.5     .05       0  4669.3      .1       0
  4959.1     .16       0    5007     .07       0    5013     .16       0
  5066.3     .05       0    5165      .1       0    5275     .05       0
  5364.2      .1       0  5498.4     .05       0  5753.8      .1       0
Bank Sta=4839.6,5030
XS Rating Curve= 0 ,0
Exp/Cntr=0.3,0.1

Type RM Length L Ch R = 1 ,59649   ,427,427,427
BEGIN DESCRIPTION:
FLAT CREEK 120.0
END DESCRIPTION:
XS GIS Cut Line= 3
      2956590.75     10049307.73      2957194.87     10049177.53
       2958528.2     10048734.82
#Sta/Elev= 30
  4118.2 1235.61  4146.6 1233.16  4161.4 1227.98    4167 1224.07  4218.2 1210.63
  4366.2 1202.07  4681.6 1189.06  4719.4 1178.67  4735.5 1171.72  4771.6 1165.05
  4826.7 1160.94  4886.6 1157.42  4971.8 1153.44  5000.4 1147.27  5003.2 1146.77
  5006.4 1147.27    5035 1153.35  5087.7 1157.05  5277.4 1170.06  5353.9 1173.58
  5472.2  1185.7    5763 1198.17    5784 1197.62  5793.7 1200.72  5810.4  1202.2
  5993.9 1214.47  6046.5 1219.92  6063.8  1218.8  6100.7 1225.65  6141.1 1228.76
#Mann= 9 ,-1 , 0
  4118.2     .05       0  4366.2      .1       0  4681.6     .05       0
  4826.7     .16       0  5000.4     .07       0  5006.4     .16       0
  5353.9      .1       0  5472.2     .05       0    5763      .1       0
Bank Sta=4886.6,5087.7
XS Rating Curve= 0 ,0
Exp/Cntr=0.3,0.1

Type RM Length L Ch R = 1 ,59222   ,731,731,731
BEGIN DESCRIPTION:
FLAT CREEK 119.0
END DESCRIPTION:
XS GIS Cut Line= 3
      2956554.27     10049427.53      2957892.79     10049521.28
      2958580.27     10049526.49
#Sta/Elev= 30
  3982.4 1236.73  4006.7 1233.39  4056.8 1219.53  4189.1 1208.91  4451.2 1196.94
  4573.8 1192.66  4719.3 1188.33  4838.7 1179.15  4888.8 1172.14  4908.9 1166.31
  4938.9 1163.21    4959 1152.52    4969 1146.87  4999.8  1145.4  5002.5  1144.9
  5005.8  1145.4  5049.2 1150.61    5060 1151.18  5189.5  1151.3    5387 1166.42
  5485.6 1176.56  5529.9 1190.76  5584.2 1190.71  5619.9 1191.83  5749.9 1205.38
  5779.9 1212.76  5835.5 1234.12  5909.9 1250.96  5978.8 1255.45  6011.7 1258.93
#Mann= 12 ,-1 , 0
  3982.4     .05       0  4189.1      .1       0  4451.2     .16       0
  4573.8      .1       0  4999.8     .07       0  5005.8      .1       0
    5060     .16       0    5387     .05       0  5485.6     .08       0
  5584.2      .1       0  5835.5     .16       0  5978.8     .05       0
#XS Ineff= 2 , 0
                         5061.36         1151.41
Permanent Ineff=
       T       T
Bank Sta=4959,5049.2
XS Rating Curve= 0 ,0
Exp/Cntr=0.3,0.1

Type RM Length L Ch R = 1 ,58491   ,639,639,639
BEGIN DESCRIPTION:
FLAT CREEK 118.0
END DESCRIPTION:
XS GIS Cut Line= 4
      2956528.22     10049516.08      2957413.62     10049932.74
      2957882.37      10050349.4      2958429.23     10050766.05
#Sta/Elev= 30
  3650.8 1233.94  3662.3 1227.67  3685.1 1222.28  3840.7 1210.93  4235.5 1188.37
  4357.2 1182.79  4466.7 1166.09  4505.1 1155.73  4556.2 1149.92  4888.8 1146.36
  4916.8 1142.33    4959 1142.46  4998.7 1135.58  5001.4 1135.08  5004.7 1135.58
  5037.2 1142.32  5101.2 1166.93  5193.2 1177.72    5256 1180.78  5285.7 1185.78
  5391.8  1187.1  5414.6 1190.12  5491.6  1185.7  5535.2  1191.4  5663.3 1199.29
  5783.4 1211.27  5805.5 1215.18  5827.9 1223.82  5869.9 1236.72    5944 1244.96
#Mann= 10 ,-1 , 0
  3650.8     .05       0  3840.7      .1       0  4235.5     .16       0
  4466.7      .1       0  4556.2     .05       0  4998.7    .035       0
  5004.7     .05       0  5663.3      .1       0  5783.4     .05       0
  5827.9      .1       0
#XS Ineff= 2 , 0
          4937.5 1143.83
Permanent Ineff=
       T       T
Bank Sta=4959,5037.2
XS Rating Curve= 0 ,0
Exp/Cntr=0.3,0.1

Type RM Length L Ch R = 1 ,57852   ,449,449,449
BEGIN DESCRIPTION:
FLAT CREEK 117.0
END DESCRIPTION:
XS GIS Cut Line= 4
      2956470.89     10049734.81      2957184.46     10050120.24
      2957200.08     10050458.78      2957903.23     10051005.67
#Sta/Elev= 30
  4004.3 1224.35  4075.5 1217.17  4275.7 1204.96  4328.4 1201.74    4438 1195.29
  4552.8 1190.13  4605.7 1185.67  4657.2 1172.23  4670.3    1169  4703.7 1153.95
  4753.2 1148.45  4850.3 1145.52  4948.9 1141.77    4969 1140.91    4979 1137.79
    4996 1131.41  4998.7 1130.91    5002 1131.41  5047.6 1134.14  5079.1 1137.82
  5146.3 1139.61  5173.2 1140.15  5390.3 1144.01  5612.4 1152.32  5648.9 1159.63
  5668.9  1166.5  5705.6 1175.27  5743.4  1179.1  5937.3 1190.92    6045 1195.49
#Mann= 19 ,-1 , 0
  4004.3     .05       0  4275.7      .1       0  4328.4     .16       0
    4438      .1       0  4552.8     .16       0  4657.2      .1       0
  4670.3     .05       0  4850.3      .1       0  4948.9     .05       0
    4996    .035       0    5002     .05       0  5047.6      .1       0
  5146.3     .05       0  5173.2      .1       0  5390.3     .05       0
  5648.9      .1       0  5668.9     .16       0  5743.4      .1       0
  5937.3     .05       0
Bank Sta=4979,5079.1
XS Rating Curve= 0 ,0
Exp/Cntr=0.3,0.1

Type RM Length L Ch R = 1 ,57403   ,650,650,650
BEGIN DESCRIPTION:
FLAT CREEK 115.0
END DESCRIPTION:
XS GIS Cut Line= 3
      2956585.46     10050505.64      2957345.92     10050766.07
      2957892.82      10051146.3
#Sta/Elev= 30
  4659.5 1220.56  4707.1 1209.58  4721.3 1205.44  4809.9 1195.21  4905.8 1178.69
  4913.5 1172.89  4918.8 1172.27  4937.5  1148.8  4944.8 1142.25  4958.6 1135.29
  4976.1 1129.84  4997.9 1126.61  5000.7 1126.11  5003.9 1126.61  5015.5 1129.58
  5032.6  1133.4  5064.3 1135.44  5118.3 1136.61  5221.1  1136.9  5304.4 1138.17
  5446.5 1141.37  5634.8 1146.24  5655.1 1147.77  5678.9 1150.52  5729.5 1169.34
  5757.5 1176.17  5765.3 1178.21  5807.4 1181.73  5989.1 1191.27  6129.4 1198.25
#Mann= 15 ,-1 , 0
  4659.5     .16       0  4707.1     .05       0  4721.3      .1       0
  4809.9     .16       0  4997.9     .07       0  5003.9     .16       0
  5015.5     .05       0  5118.3      .1       0  5221.1     .05       0
  5304.4      .1       0  5446.5     .05       0  5634.8      .1       0
  5655.1     .16       0  5757.5      .1       0  5989.1     .05       0
Bank Sta=4958.6,5064.3
XS Rating Curve= 0 ,0
Exp/Cntr=0.3,0.1

Type RM Length L Ch R = 1 ,56753   ,542,542,542
BEGIN DESCRIPTION:
FLAT CREEK 114.0
END DESCRIPTION:
XS GIS Cut Line= 4
      2956246.96     10051026.49      2956627.17     10051266.07
       2957085.5     10051240.03      2957823.04     10051749.04
#Sta/Elev= 30
  4315.7 1261.81  4394.6 1238.41  4485.2 1224.53  4518.4 1219.45  4553.9 1206.56
    4583 1202.12  4619.5  1186.8  4659.3 1177.12  4671.2 1171.74  4677.1 1172.86
  4692.4  1161.4  4698.3 1161.92  4713.6 1152.27  4732.5 1149.38  4776.4 1139.26
  4835.7  1134.4  4946.7 1129.76  4993.8 1120.06  4996.5 1119.56  4999.8 1120.06
  5033.8 1126.78  5046.8 1129.33  5167.6 1132.21  5337.1 1141.95  5466.3 1155.72
  5609.9 1164.98    5687 1175.36  5728.4 1179.89  5877.8 1189.87  6120.3 1204.06
#Mann= 13 ,-1 , 0
  4315.7     .16       0  4485.2     .05       0  4659.3     .16       0
  4732.5      .1       0  4835.7     .16       0  4993.8     .07       0
  4999.8     .16       0  5033.8      .1       0  5167.6     .05       0
  5466.3      .1       0    5687     .16       0  5728.4      .1       0
  5877.8     .05       0
Bank Sta=4946.7,5046.8
XS Rating Curve= 0 ,0
Exp/Cntr=0.3,0.1

Type RM Length L Ch R = 1 ,56211   ,380,380,380
BEGIN DESCRIPTION:
FLAT CREEK 113.0
END DESCRIPTION:
XS GIS Cut Line= 2
      2956189.66     10051130.65        2957361.     10052359.26
#Sta/Elev= 30
  4139.3 1254.72  4161.8 1250.57  4211.5 1233.85  4263.8 1225.13    4275 1220.41
  4296.1 1217.55  4317.5 1211.31  4388.3 1205.91  4442.7 1196.92  4501.5 1181.22
  4582.7 1151.82  4621.6 1141.62  4699.3 1132.26  4805.6 1126.66  4954.1 1124.77
  4993.6 1116.96  4996.3 1116.46  4999.6 1116.96  5017.6 1119.02  5031.8 1124.07
  5045.9  1129.1  5152.3 1134.53  5212.9 1138.25  5364.8  1147.5  5407.8    1151
  5526.8 1157.46  5604.8 1170.46  5673.1 1177.12    5810 1184.26  5836.8 1186.15
#Mann= 12 ,-1 , 0
  4139.3     .16       0  4263.8      .1       0  4442.7     .16       0
  4582.7     .05       0  4993.6    .035       0  4999.6     .05       0
  5152.3      .1       0  5212.9     .05       0  5364.8      .1       0
  5407.8     .16       0  5673.1      .1       0    5810     .05       0
Bank Sta=4954.1,5031.8
XS Rating Curve= 0 ,0
Exp/Cntr=0.3,0.1

Type RM Length L Ch R = 1 ,55831   ,580,580,580
BEGIN DESCRIPTION:
FLAT CREEK 112.0
END DESCRIPTION:
XS GIS Cut Line= 3
       2955851.1     10051516.06      2956345.92      10051849.4
      2957053.86     10052567.76
#Sta/Elev= 30
  4160.6 1236.86  4164.4 1233.13  4193.6 1223.63  4221.4 1221.17  4272.4 1210.22
  4302.1 1207.73  4365.3 1198.26  4398.4 1188.91  4416.3 1185.61  4437.3 1177.74
  4518.2 1157.11  4560.2 1150.51  4634.3 1144.35  4945.9 1123.73  4953.9 1122.31
  4999.5 1112.83  5002.2 1112.33  5005.5 1112.83  5016.6 1116.71  5080.3 1122.47
  5165.2 1125.43  5242.9 1132.05  5275.4 1133.12  5338.3 1137.22    5494 1151.34
  5575.3 1163.37  5596.5 1164.58  5617.7 1170.24  5677.8 1177.11  5765.8 1183.55
#Mann= 10 ,-1 , 0
  4160.6     .16       0  4398.4      .1       0  4634.3     .05       0
  4953.9     .16       0  4999.5     .07       0  5005.5     .16       0
  5275.4     .05       0  5338.3      .1       0    5494     .16       0
  5677.8      .1       0
Bank Sta=4945.9,5080.3
XS Rating Curve= 0 ,0
Exp/Cntr=0.3,0.1

Type RM Length L Ch R = 1 ,55251   ,541,541,541
BEGIN DESCRIPTION:
FLAT CREEK 111.0
END DESCRIPTION:
XS GIS Cut Line= 2
      2955621.94     10051844.17      2956647.21     10052999.56
#Sta/Elev= 30
  4125.5  1211.9  4313.7 1197.74  4378.1 1189.03  4448.3 1182.47  4462.5 1178.81
  4476.8 1172.53  4519.4 1147.51  4556.6 1133.89  4576.3 1129.27  4618.9 1124.25
  4754.1 1121.24  4927.3 1117.21  4937.6 1117.45  4980.2 1115.14  4998.1 1108.97
  5000.9 1108.47  5004.1 1108.97  5015.3 1113.56  5043.8 1119.06  5069.2 1121.44
  5103.1 1123.58    5211 1129.66  5239.8 1131.37  5352.9 1138.58  5376.4 1140.65
    5426 1147.26  5468.6 1156.53    5537 1167.72    5610 1179.33  5670.2 1184.49
#Mann= 13 ,-1 , 0
  4125.5     .16       0  4556.6     .05       0  4754.1      .1       0
  4927.3     .16       0  4998.1     .07       0  5004.1     .16       0
  5069.2     .05       0  5103.1      .1       0    5211     .05       0
  5239.8      .1       0  5352.9     .16       0  5376.4      .1       0
    5537     .05       0
Bank Sta=4937.6,5043.8
XS Rating Curve= 0 ,0
Exp/Cntr=0.3,0.1

Type RM Length L Ch R = 1 ,54710   ,478,478,478
BEGIN DESCRIPTION:
FLAT CREEK 110.0
END DESCRIPTION:
XS GIS Cut Line= 3
      2955486.54      10051719.2      2955804.25     10052990.03
      2956361.52     10053234.81
#Sta/Elev= 30
  3948.3 1236.71  3972.6 1229.62  3977.8  1232.5  4004.5 1220.84    4019 1219.94
  4025.1 1216.35  4045.7 1211.68  4170.2 1206.45  4251.9 1199.29  4348.9 1185.37
  4390.1 1174.64  4437.4 1152.63  4467.4 1141.54  4498.3 1134.22  4549.9 1127.58
  4643.6 1120.95  4816.2 1115.74  4973.4 1111.26  5005.6 1107.04  5008.3 1106.54
  5011.6 1107.04  5044.6 1111.57  5074.6 1118.57  5107.4 1126.35  5310.8  1132.3
  5524.7 1145.08  5622.9 1148.38  5714.3 1156.35  5756.1  1162.9  5866.9  1171.2
#Mann= 10 ,-1 , 0
  3948.3      .1       0  4170.2     .16       0  4498.3     .05       0
  4816.2      .1       0  5005.6     .07       0  5011.6      .1       0
  5074.6     .05       0  5310.8      .1       0  5524.7     .05       0
  5714.3      .1       0
Bank Sta=4973.4,5044.6
XS Rating Curve= 0 ,0
Exp/Cntr=0.3,0.1

Type RM Length L Ch R = 1 ,54232   ,392,392,392
BEGIN DESCRIPTION:
FLAT CREEK 109.0
END DESCRIPTION:
XS GIS Cut Line= 4
      2954476.11     10052266.06      2955215.71     10052818.15
      2955486.54      10053099.4      2956299.07     10053271.29
#Sta/Elev= 30
  3951.2 1212.02  4016.1 1208.87  4122.7 1203.14  4408.3 1199.81    4473 1193.52
  4615.5 1186.01  4679.3 1174.86    4744 1156.13  4758.6 1150.71  4787.8 1133.31
  4808.6 1125.49  4815.2 1120.67  4885.2 1111.47  4922.6 1108.64  4979.1 1106.45
  4990.1 1102.52  4992.8 1102.02  4996.1 1102.52  5021.4 1106.69    5071 1109.54
  5111.2 1113.09  5205.3 1118.98  5353.7 1123.51    5450 1129.27  5593.6 1133.71
  5739.8 1143.91  5920.7 1153.02  6012.6 1161.61  6057.8 1165.41  6095.1 1167.42
#Mann= 10 ,-1 , 0
  3951.2      .1       0  4016.1     .16       0  4885.2     .05       0
  4990.1    .035       0  4996.1     .05       0  5111.2     .16       0
  5353.7      .1       0  5739.8     .05       0  6012.6      .1       0
  6057.8     .16       0
Bank Sta=4922.6,5071
XS Rating Curve= 0 ,0
Exp/Cntr=0.3,0.1

Type RM Length L Ch R = 1 ,53840   ,492,492,492
BEGIN DESCRIPTION:
FLAT CREEK 108.0
END DESCRIPTION:
XS GIS Cut Line= 3
      2954616.75     10052854.61      2954804.25      10053156.7
      2956283.42     10053375.45
#Sta/Elev= 30
  4338.4 1197.53  4368.4  1193.2  4389.7  1195.3  4405.1 1192.89  4447.6 1195.65
  4462.9 1194.23  4484.2 1197.56  4499.5 1194.78  4599.9 1195.01  4705.6 1188.71
  4839.6 1163.65  4900.4 1139.28  4914.2 1130.95  4920.6 1122.59  4930.7 1115.09
  4950.9 1104.96  4998.5 1097.28  5001.2 1096.78  5004.5 1097.28  5028.4 1102.18
  5048.3 1106.85  5313.3 1114.87    5426 1119.53  5466.5 1125.08  5546.1 1129.69
  5688.9 1134.38  5786.2 1140.55  6019.6 1151.36  6068.2 1161.03  6189.2 1168.11
#Mann= 9 ,-1 , 0
  4338.4     .16       0  4998.5     .07       0  5004.5     .16       0
  5028.4     .05       0  5313.3     .16       0  5546.1      .1       0
  5786.2     .05       0  6019.6      .1       0  6068.2     .16       0
Bank Sta=4950.9,5048.3
XS Rating Curve= 0 ,0
Exp/Cntr=0.3,0.1

Type RM Length L Ch R = 1 ,53348   ,499,499,499
BEGIN DESCRIPTION:
FLAT CREEK 107.0
END DESCRIPTION:
XS GIS Cut Line= 4
      2954475.34     10053509.77      2954851.71     10053684.52
      2955379.27      10053694.6      2955854.93     10053862.08
#Sta/Elev= 30
  4377.5 1181.25  4436.9 1176.35  4543.5 1159.18  4564.4 1152.84  4609.7 1145.17
  4650.2 1142.11  4756.9 1136.63  4792.5 1130.56  4809.2 1123.23  4839.2 1122.64
  4858.2 1118.59  4919.2 1112.95 4943.52 1103.43  4949.2 1100.37  4979.3 1098.95
  4996.3 1094.47    4999 1093.97  5002.3 1094.47  5029.3  1099.6  5129.3 1103.36
  5359.5 1112.24  5382.9 1106.26  5435.9 1117.67  5452.4 1124.61  5520.7  1131.4
  5598.9 1133.01  5720.4 1139.49  5787.6 1139.78  5809.9 1144.47  5824.4 1146.56
#Mann= 11 ,-1 , 0
  4377.5      .1       0  4436.9     .05       0  4543.5      .1       0
  4564.4     .05       0  4650.2     .16       0  4756.9      .1       0
  4858.2     .16       0  4996.3     .07       0  5002.3     .16       0
  5598.9     .05       0  5809.9      .1       0
#XS Ineff= 2 , 0
                            5280         1110.94
Permanent Ineff=
       T       T
Bank Sta=4943.52,5129.3
XS Rating Curve= 0 ,0
Exp/Cntr=0.3,0.1

Type RM Length L Ch R = 1 ,52849   ,658,658,658
BEGIN DESCRIPTION:
FLAT CREEK 106.0
END DESCRIPTION:
XS GIS Cut Line= 4
        2954472.     10053610.58      2954915.56     10054070.94
      2955103.73     10054242.31      2955424.85     10054372.77
#Sta/Elev= 30
    4204 1176.45  4267.3 1168.99  4288.7 1163.71  4309.8 1161.59  4345.3 1152.84
  4352.2 1153.81  4380.5 1149.75  4446.2 1145.92  4557.2  1136.8  4585.5 1129.61
  4606.9 1120.86  4656.3 1109.28  4663.5  1105.4  4687.1 1101.59    4731 1099.65
  4823.2 1098.45  4932.1 1099.57  4960.5 1096.54    4993 1089.49  4995.7 1088.99
    4999 1089.49  5045.6 1095.15    5117 1099.21  5135.3 1103.33  5146.4 1109.37
  5194.6 1120.73  5210.8 1127.07  5293.7 1133.74  5398.4 1137.31  5444.4 1139.98
#Mann= 9 ,-1 , 0
    4204     .05       0  4446.2     .16       0  4687.1     .05       0
    4731      .1       0  4823.2     .16       0    4993     .07       0
    4999     .16       0  5293.7     .05       0  5398.4     .08       0
#XS Ineff= 1 ,-1
 4695.91  4925.4 1100.21
Permanent Ineff=
       T
Bank Sta=4932.1,5117
XS Rating Curve= 0 ,0
Exp/Cntr=0.3,0.1

Type RM Length L Ch R = 1 ,52191   ,410,410,410
BEGIN DESCRIPTION:
FLAT CREEK 105.0
END DESCRIPTION:
XS GIS Cut Line= 4
      2954361.12     10053597.16      2954445.13     10053916.37
      2954465.29     10054302.79      2955065.12     10054527.31
#Sta/Elev= 30
  4422.1 1182.31  4532.3 1170.99  4563.3 1163.49  4588.8 1161.57    4624 1154.38
  4656.4 1150.87  4664.3 1147.81  4739.1 1138.61  4752.2 1135.21  4809.5 1109.84
  4849.7 1099.02  4901.9    1095  4929.8 1093.48  4979.8 1088.55  4996.9  1083.5
  4999.6    1083  5002.9  1083.5  5019.9 1089.47    5090 1093.32    5172 1095.65
  5323.2 1100.34  5508.9 1107.27  5569.6 1108.88  5645.4 1117.92  5664.4 1118.71
  5695.2 1121.07  5719.1 1125.64  5730.9 1130.05  5775.9 1131.45  5779.6 1131.43
#Mann= 10 ,-1 , 0
  4422.1     .16       0  4809.5     .05       0  4901.9     .16       0
  4996.9     .07       0  5002.9     .16       0    5172      .1       0
  5323.2     .16       0  5508.9     .05       0  5664.4      .1       0
  5775.9     .05       0
Bank Sta=4929.8,5090
XS Rating Curve= 0 ,0
Exp/Cntr=0.3,0.1

Type RM Length L Ch R = 1 ,51781   ,395,395,395
BEGIN DESCRIPTION:
FLAT CREEK 103.0
END DESCRIPTION:
XS GIS Cut Line= 3
      2953158.17     10054158.31      2954535.85       10054454.
      2955049.96     10054548.09
#Sta/Elev= 30
  3983.1 1155.62  4382.3 1143.99  4678.9 1138.39  4751.6 1132.97  4790.7 1122.63
  4852.8 1120.32  4883.4 1113.06  4889.5 1109.92  4924.4  1102.4  4933.8 1099.45
  4945.8  1093.6    4955 1089.03  4992.9 1081.21  4995.7 1080.71  4998.9 1081.21
  5045.8 1088.11  5067.5  1090.5  5118.7 1092.89  5145.8 1092.73  5245.8 1094.24
  5345.8 1096.57  5457.6 1100.14  5530.8 1102.73  5634.4 1108.54  5689.6 1112.51
    5710 1116.02  5791.3 1120.22  5865.2 1131.98  5914.2 1132.37  5914.8 1132.37
#Mann= 11 ,-1 , 0
  3983.1     .16       0  4945.8     .05       0  4992.9    .035       0
  4998.9     .05       0  5045.8      .1       0  5145.8     .05       0
  5245.8     .16       0  5345.8      .1       0  5457.6     .16       0
  5634.4      .1       0  5914.2     .05       0
#XS Ineff= 2 ,-1
 5175.53  5211.6    1093 5269.09 5288.34 1095.44
Permanent Ineff=
       T       T
Bank Sta=4955,5067.5
XS Rating Curve= 0 ,0
Exp/Cntr=0.3,0.1
