HEC-RAS study MILLER CREEK.prj: MILLER CREEK Base Level Engineering

--- MILLER CREEK.g01 (geometry) --- (continued)

Type RM Length L Ch R = 1 ,101851  ,766,766,766
BEGIN DESCRIPTION:
MILLER CREEK 162.0
END DESCRIPTION:
XS GIS Cut Line= 4
      2903578.28     10043972.42      2904251.88     10042444.66
       2904661.6     10041847.44      2904515.76     10040861.29
#Sta/Elev= 30
  2843.1 1383.72  2880.1 1382.85  3228.7 1375.49  3311.6  1368.3  3350.8 1359.73
  3426.2 1354.54  3496.2 1343.05  3552.3 1339.72  4351.1 1318.71  4456.6 1316.67
  4864.3  1310.9  4971.9 1305.53  4986.8 1299.09  5004.8 1298.84  5007.5 1298.34
  5010.8 1298.84  5043.6 1312.12  5085.6  1319.6  5125.3 1319.08  5498.1 1319.81
  5562.6 1324.21    5616 1332.74  5695.7 1359.57  5776.5 1405.02  5827.1 1425.26
  5857.4  1450.1  5883.7 1452.92  6115.8 1467.76  6159.5  1471.9  6233.9 1478.28
#Mann= 12 ,-1 , 0
  2843.1     .05       0  2880.1      .1       0  3552.3     .05       0
  4351.1      .1       0  4456.6     .05       0  5004.8    .035       0
  5010.8     .05       0  5125.3      .1       0    5616     .16       0
  5883.7      .1       0  6115.8     .05       0  6159.5      .1       0
#XS Ineff= 4 ,-1
 4492.21 4531.41 1315.57 4533.08 4655.71 1314.85  4677.4 4719.94 1314.85
 5095.33  6233.9 1320.05
Permanent Ineff=
       T       T       T       T
Bank Sta=4864.3,5043.6
XS Rating Curve= 0 ,0
Exp/Cntr=0.3,0.1

Type RM Length L Ch R = 1 ,101085  ,1137,1137,1137
BEGIN DESCRIPTION:
MILLER CREEK 161.0
END DESCRIPTION:
XS GIS Cut Line= 4
      2904411.58     10044111.37      2905140.77     10042944.66
      2905133.82     10041972.44      2904543.54     10040784.94
#Sta/Elev= 30
  3120.8 1368.71  3159.5 1368.13  3272.5 1365.29  3498.5 1354.87  3554.9 1350.58
  3789.4  1337.3  4161.9  1326.3  4808.2 1324.43  4907.6  1318.9  4947.6 1309.56
  4977.6 1299.45  5004.6    1299  5007.3  1298.5  5010.6    1299    5020 1299.39
  5103.4 1306.87  5117.6 1308.72  5576.9 1316.62  5696.2 1316.83  5837.6 1317.39
  5948.4 1317.98  6182.1  1334.1  6277.8 1385.75  6350.5 1409.12  6389.8 1409.89
  6434.6 1419.82  6484.9 1448.06  6580.9 1457.89  6623.1 1460.84    6795  1481.2
#Mann= 17 ,-1 , 0
  3120.8      .1       0  3159.5     .05       0  3272.5      .1       0
  3498.5     .05       0  3554.9      .1       0  3789.4     .05       0
  4808.2      .1       0  5004.6     .07       0  5010.6      .1       0
    5020     .05       0  5103.4      .1       0  5576.9     .05       0
  5696.2      .1       0  5837.6     .05       0  5948.4     .16       0
  6580.9      .1       0  6623.1     .05       0
Bank Sta=4947.6,5117.6
XS Rating Curve= 0 ,0
Exp/Cntr=0.3,0.1

Type RM Length L Ch R = 1 ,99948   ,923,923,923
BEGIN DESCRIPTION:
MILLER CREEK 159.0
END DESCRIPTION:
XS GIS Cut Line= 3
      2904841.92      10044184.4      2905939.12     10042608.05
      2906175.23     10041330.29
#Sta/Elev= 30
  2364.6 1347.81  2387.9 1347.46  2577.7 1341.99  2641.5 1339.03  2692.1 1337.46
    2827  1333.2  3003.6 1326.91  3220.4  1322.3    3284 1322.33  3404.4 1319.01
  3516.8 1317.54  3588.4 1316.16  3633.2 1315.47  3840.2 1313.62  4517.5 1309.74
  4750.9 1308.84  4828.6 1302.49  4861.8 1299.11  4998.5  1288.8  5001.2  1288.3
  5004.5  1288.8    5032 1303.47  5072.6 1318.44  5112.2 1341.68    5154    1371
  5189.6 1388.47  5225.2 1399.37  5316.7  1441.3  5439.6 1446.08  5584.6 1448.23
#Mann= 20 ,-1 , 0
  2364.6     .05       0  2387.9      .1       0  2577.7     .05       0
  2641.5      .1       0  2692.1     .05       0    2827      .1       0
  3003.6     .05       0  3220.4      .1       0    3284     .05       0
  3404.4      .1       0  3516.8     .05       0  3588.4      .1       0
  3633.2     .05       0  3840.2     .05       0  4517.5     .05       0
  4861.8      .1       0  4998.5     .07       0  5004.5      .1       0
  5112.2     .16       0  5439.6      .1       0
Bank Sta=4828.6,5032
XS Rating Curve= 0 ,0
Exp/Cntr=0.3,0.1

Type RM Length L Ch R = 1 ,99025   ,605,605,605
BEGIN DESCRIPTION:
MILLER CREEK 158.0
END DESCRIPTION:
XS GIS Cut Line= 4
       2905529.4     10043392.77      2906508.56      10042788.6
       2906841.9     10042364.99      2906459.97     10041392.81
#Sta/Elev= 30
  3556.6 1318.61  3616.1 1317.39  3624.6 1316.96    3917 1313.36  4393.1 1309.55
  4623.2 1305.26  4745.5 1301.41  4826.7 1300.27  4916.9 1295.83  4947.8 1291.69
  4999.9 1286.41  5002.7 1285.91  5005.9 1286.41  5081.5 1295.47  5135.5 1300.74
    5190 1303.26  5488.7 1315.76  5537.5  1323.4  5580.6 1335.41  5621.5 1339.86
  5656.7 1349.93  5675.7 1349.57  5733.8 1362.03  5784.1  1365.3  5981.9 1390.13
  6090.3 1389.94  6114.7 1383.19    6169 1380.55  6252.8 1382.66  6290.7 1390.17
#Mann= 15 ,-1 , 0
  3556.6      .1       0  3616.1     .05       0  3624.6      .1       0
    3917     .05       0  4393.1      .1       0  4623.2     .05       0
  4745.5      .1       0  4826.7     .05       0  4947.8      .1       0
  4999.9     .07       0  5005.9      .1       0  5135.5     .05       0
    5190      .1       0  5733.8     .05       0  6252.8      .1       0
Bank Sta=4916.9,5081.5
XS Rating Curve= 0 ,0
Exp/Cntr=0.3,0.1

Type RM Length L Ch R = 1 ,98420   ,718,718,718
BEGIN DESCRIPTION:
MILLER CREEK 157.0
END DESCRIPTION:
XS GIS Cut Line= 3
      2907008.83     10044166.85      2907133.82     10043055.77
      2907418.19     10041536.84
#Sta/Elev= 30
  3720.2 1351.26  4092.8 1331.83  4357.3  1317.5  4596.7 1308.89  4810.1 1302.81
  4833.6 1299.23  4931.9 1291.66  4995.7 1279.98  4998.5 1279.48  5001.7 1279.98
  5033.7 1281.99  5047.5 1285.99    5115  1291.9  5160.6 1297.49  5371.6 1300.73
  5470.2 1300.46  5572.9 1300.27  5597.7 1304.18  5633.9 1297.92  5664.4 1304.13
  5708.5 1302.72  5959.5 1312.48  6061.2  1319.9  6132.4 1333.04  6213.8 1360.88
  6244.2 1363.61  6264.7 1369.81  6325.7 1371.49  6359.6 1377.86  6383.6 1378.61
#Mann= 11 ,-1 , 0
  3720.2      .1       0  4092.8     .05       0  4596.7      .1       0
  4833.6     .05       0  4995.7    .035       0  5001.7     .05       0
  5047.5      .1       0  5160.6     .05       0  5371.6      .1       0
  5470.2     .05       0  5708.5      .1       0
#XS Ineff= 2 , 0
                         5324.48         1300.91
Permanent Ineff=
       T       T
Bank Sta=4931.9,5115
XS Rating Curve= 0 ,0
Exp/Cntr=0.3,0.1

Type RM Length L Ch R = 1 ,97702   ,715,715,715
BEGIN DESCRIPTION:
MILLER CREEK 156.0
END DESCRIPTION:
XS GIS Cut Line= 4
      2907453.27     10044159.91       2907849.1       10042653.
      2907383.82     10042048.83      2907675.48     10041340.53
#Sta/Elev= 30
  3226.8 1346.93  3379.6  1338.6  3616.5 1325.91  3794.1 1315.95  3953.4 1309.44
  4291.6 1300.54  4688.7 1301.43  4707.9 1300.55  4788.5 1298.03  4810.3 1296.61
  4891.8 1286.92  4995.5 1274.72  4998.2 1274.22  5001.5 1274.72  5012.3 1275.56
    5035 1287.61  5058.4 1291.75  5234.3 1290.24  5301.9 1296.71  5651.6 1311.84
  5706.9 1314.78  5741.6 1322.26  5784.1 1333.04  5808.1 1346.11  5861.4 1364.28
    5907 1374.24  5985.5 1386.05  6074.6 1414.13  6177.3  1427.7  6313.4 1428.69
#Mann= 17 ,-1 , 0
  3226.8      .1       0  3379.6     .05       0  3616.5      .1       0
  3794.1     .05       0  3953.4      .1       0  4688.7     .05       0
  4707.9      .1       0  4788.5     .05       0  4810.3      .1       0
  4995.5     .07       0  5001.5      .1       0  5058.4     .05       0
  5301.9      .1       0  5651.6     .05       0  5741.6      .1       0
    5907     .16       0  6177.3      .1       0
#XS Ineff= 2 , 0
                         5139.77         1294.69
Permanent Ineff=
       T       T
Bank Sta=4891.8,5035
XS Rating Curve= 0 ,0
Exp/Cntr=0.3,0.1

Type RM Length L Ch R = 1 ,96987   ,1212,1212,1212
BEGIN DESCRIPTION:
MILLER CREEK 154.0
END DESCRIPTION:
XS GIS Cut Line= 4
      2907640.75     10044083.59      2908307.43     10042368.27
      2908342.16     10041909.94        2908155.     10041417.79
#Sta/Elev= 30
  2924.1 1341.39  2992.9 1337.73  3023.9 1336.35  3096.7 1332.76  3340.4 1317.61
  3494.4 1308.92  3943.2 1293.15  3982.9 1297.55  4134.8 1295.31  4362.7 1294.56
  4579.5 1290.74  4809.1 1284.09  4996.6 1272.74  4999.4 1272.24  5002.6 1272.74
  5039.8 1283.93  5053.1  1291.3  5069.8 1300.18    5140 1310.59  5185.3 1323.54
  5247.6  1351.4    5253 1349.49  5272.4  1361.2  5277.8 1358.88  5302.5 1374.51
  5412.3 1384.76  5471.1 1403.91  5532.7 1416.43  5642.5 1427.69  5750.6 1431.56
#Mann= 15 ,-1 , 0
  2924.1      .1       0  2992.9     .05       0  3023.9     .16       0
  3096.7     .05       0  3340.4      .1       0  3494.4     .05       0
  3982.9      .1       0  4134.8     .05       0  4362.7      .1       0
  4579.5     .05       0  4996.6     .04       0  5002.6     .05       0
  5053.1      .1       0  5185.3     .16       0  5471.1      .1       0
#XS Ineff= 3 ,-1
 3911.38 3975.33 1296.34 4128.95 4189.91 1295.77 4221.59 4264.03 1294.13
Permanent Ineff=
       T       T       T
Bank Sta=4809.1,5039.8
XS Rating Curve= 0 ,0
Exp/Cntr=0.3,0.1

Type RM Length L Ch R = 1 ,95775   ,595,595,595
BEGIN DESCRIPTION:
MILLER CREEK 152.0
END DESCRIPTION:
XS GIS Cut Line= 4
      2909224.11     10044486.36      2908835.21     10043430.77
      2909071.32     10041979.38      2908987.99     10041021.01
#Sta/Elev= 30
  3521.7 1338.24  3647.9 1333.33  3704.6 1331.61  4090.5 1321.42  4210.9 1317.71
  4424.8 1309.32  4775.4 1304.51  4917.2 1292.52  4927.3  1290.5 4940.91 1281.43
  4967.9 1269.75  5008.4 1266.69  5011.2 1266.19  5014.4 1266.69  5129.4 1281.38
  5190.7 1287.81  5260.8 1287.88  5501.5  1291.3  6152.9 1300.62  6413.9 1312.48
  6556.8 1331.52  6634.7 1353.92  6694.9  1366.2  6735.1 1366.55  6835.5 1378.97
  6925.8 1384.18  7013.5 1406.73  7018.5 1404.34  7073.1 1415.53  7079.1 1415.77
#Mann= 11 ,-1 , 0
  3521.7      .1       0  3647.9     .16       0  3704.6      .1       0
  4090.5     .16       0  4210.9     .05       0  4424.8      .1       0
  5008.4     .07       0  5014.4      .1       0  5260.8     .05       0
  5501.5      .1       0  7073.1     .16       0
Bank Sta=4940.91,5129.4
XS Rating Curve= 0 ,0
Exp/Cntr=0.3,0.1

Type RM Length L Ch R = 1 ,95180   ,630,630,630
BEGIN DESCRIPTION:
MILLER CREEK 151.0
END DESCRIPTION:
XS GIS Cut Line= 4
      2909696.31     10044277.96      2909446.32     10043639.11
       2909474.1       10042403.      2909029.69     10040958.66
#Sta/Elev= 30
  3660.7 1344.48  3867.8 1340.24  4063.3 1331.33  4170.8 1325.76  4382.3 1319.14
  4612.2 1310.66  4782.2 1295.23  4832.2 1287.23  4842.2 1279.53  4922.2 1274.81
  4999.3 1259.36    5002 1258.86  5005.3 1259.36  5032.3  1276.7  5052.3 1279.94
  5070.4 1282.31  5463.6 1288.62  5538.8  1288.2  5698.2 1288.02  5714.9 1287.98
  5857.6 1288.53  6290.5 1298.74    6328 1301.71  6422.7  1310.2  6555.4 1330.55
  6644.2 1357.65  6848.5 1382.34  6932.1 1410.69  6979.7 1416.11  7094.3 1427.54
#Mann= 18 ,-1 , 0
  3660.7     .16       0  3867.8      .1       0  4063.3     .05       0
  4170.8      .1       0  4382.3     .16       0  4999.3     .07       0
  5005.3     .16       0  5070.4     .05       0  5463.6      .1       0
  5538.8     .05       0  5698.2      .1       0  5714.9     .05       0
  5857.6      .1       0  6290.5     .16       0    6328      .1       0
  6422.7     .16       0  6644.2      .1       0  6979.7     .16       0
#XS Ineff= 1 ,-1
 5112.17 5202.48 1285.71
Permanent Ineff=
       T
Bank Sta=4842.2,5052.3
XS Rating Curve= 0 ,0
Exp/Cntr=0.3,0.1

Type RM Length L Ch R = 1 ,94550   ,374,374,374
BEGIN DESCRIPTION:
MILLER CREEK 150.0
END DESCRIPTION:
XS GIS Cut Line= 4
      2910404.66     10043812.71      2910307.43      10043215.5
      2909543.55     10042104.38      2909286.61     10041000.23
#Sta/Elev= 30
  3937.3 1338.44  4008.8 1337.33    4291 1326.46  4681.8 1299.41  4866.6 1295.41
  4902.5 1287.46  4921.4 1275.78  4993.5 1259.61    5007 1259.28  5009.8 1258.78
    5013 1259.28  5102.7  1275.6    5184  1283.3  5343.9 1287.13  5487.3 1286.76
  5561.6 1286.43  5601.8  1286.3  5733.1 1286.19  5867.7 1286.45  5928.6 1286.88
  5963.9  1286.7  6296.4  1291.5  6497.2 1299.39  6589.6 1320.35  6676.9 1357.97
  6743.6 1372.03  6825.7 1377.75  6904.3 1410.89  6979.7 1411.37  7024.4 1417.25
#Mann= 19 ,-1 , 0
  3937.3     .05       0  4008.8     .16       0    4291      .1       0
  4681.8     .16       0  4921.4      .1       0  4993.5     .16       0
    5007     .07       0    5013     .16       0    5184     .05       0
  5343.9      .1       0  5487.3     .05       0  5561.6      .1       0
  5601.8     .05       0  5733.1      .1       0  5867.7     .05       0
  5928.6      .1       0  5963.9     .05       0  6296.4     .16       0
  6676.9      .1       0
Bank Sta=4921.4,5102.7
XS Rating Curve= 0 ,0
Exp/Cntr=0.3,0.1

Type RM Length L Ch R = 1 ,94176   ,1544,1544,1544
BEGIN DESCRIPTION:
MILLER CREEK 149.0
END DESCRIPTION:
XS GIS Cut Line= 4
      2910460.21     10043152.96      2910446.32     10042659.94
      2909967.16     10042347.44      2909689.39     10040923.87
#Sta/Elev= 30
  4277.3 1317.54  4519.3 1312.46  4706.7 1301.45  4851.7 1286.35  4875.3 1275.96
    4882 1273.64  4939.3 1269.06  4969.5 1260.47  4987.6 1259.11  4990.4 1258.61
  4993.6 1259.11  5018.7 1260.77  5055.1 1270.81    5069 1272.91  5156.6 1283.48
    5227 1285.58  5747.3 1283.47  6177.3 1282.42  6352.3 1283.11    6400 1285.82
  6446.7 1293.91  6460.2 1298.83  6506.7 1321.87    6518 1330.61  6558.3 1352.71
    6569 1364.22  6579.2 1368.68    6620 1370.89  6701.4 1365.04    6793 1362.93
#Mann= 10 ,-1 , 0
  4277.3      .1       0  4875.3     .16       0  4987.6     .07       0
  4993.6     .16       0  5055.1     .05       0    5227      .1       0
  5747.3     .05       0  6177.3      .1       0  6352.3     .05       0
    6400     .16       0
#XS Ineff= 2 , 0
                         5261.36         1285.21
Permanent Ineff=
       T       T
Bank Sta=4882,5069
XS Rating Curve= 0 ,0
Exp/Cntr=0.3,0.1

Type RM Length L Ch R = 1 ,92632   ,739,739,739
BEGIN DESCRIPTION:
MILLER CREEK 146.0
END DESCRIPTION:
XS GIS Cut Line= 3
      2910515.76     10043208.59      2910862.99     10041548.83
      2910460.22     10040791.91
#Sta/Elev= 30
  2844.1 1319.09  3070.8 1315.23  3227.9 1310.26  3398.3 1298.74  3625.5 1288.92
  3792.6 1288.26  4106.7 1288.91  4561.3 1274.65  4650.9 1268.47  4738.1 1263.32
  4780.1 1261.68  4824.7 1261.33  4895.9 1260.79  4974.6 1253.54  4983.8 1247.39
  4995.7 1245.47  4998.4 1244.97  5001.7 1245.47  5021.3 1248.23    5044 1261.26
 5044.89 1264.48  5055.3 1275.78    5066 1279.33  5137.6 1286.15  5191.2 1297.64
  5236.1 1309.34  5270.5 1325.86  5285.7 1329.83  5329.6  1339.4  5397.2 1341.36
#Mann= 10 ,-1 , 0
  2844.1      .1       0  3070.8     .05       0  3398.3      .1       0
  3792.6     .05       0  4650.9      .1       0  4780.1     .05       0
  4824.7      .1       0  4974.6     .16       0  4995.7     .07       0
  5001.7     .16       0
Bank Sta=4738.1,5044.89
XS Rating Curve= 0 ,0
Exp/Cntr=0.3,0.1

Type RM Length L Ch R = 1 ,91893   ,878,878,878
BEGIN DESCRIPTION:
MILLER CREEK 145.0
END DESCRIPTION:
XS GIS Cut Line= 3
      2910592.16     10043215.49      2911182.43      10041215.5
       2912008.8     10039764.15
#Sta/Elev= 30
    2634 1319.78  3007.5 1307.68  3155.8  1299.3  3524.5 1277.39  3602.3 1283.61
  3906.1 1281.39    4334  1272.7  4537.8 1267.55  4716.4 1263.92  4804.9 1260.25
  4826.7 1258.89  4907.2 1253.62  4937.2 1255.52  4984.9 1245.02  4987.7 1244.52
  4990.9 1245.02  5008.7 1245.29  5084.5 1260.83  5106.1 1267.97  5165.2 1267.11
    5230 1278.69  5348.3 1284.27  5658.3 1297.18  5745.5 1299.73  6133.5 1357.03
  6205.5 1360.72  6254.6 1367.65  6309.3 1391.53  6359.8 1395.72  6389.4 1402.92
#Mann= 17 ,-1 , 0
    2634      .1       0  3007.5     .05       0  3155.8      .1       0
  3602.3     .16       0  3906.1      .1       0    4334     .05       0
  4537.8      .1       0  4716.4     .05       0  4826.7     .16       0
  4937.2     .05       0  4984.9    .035       0  4990.9     .05       0
  5008.7     .16       0  5348.3      .1       0  5658.3     .16       0
  6205.5      .1       0  6254.6     .16       0
#XS Ineff= 2 ,-1
    2634 4599.43 1269.06 5127.76 5191.52 1269.39
Permanent Ineff=
       T       T
Bank Sta=4804.9,5084.5
XS Rating Curve= 0 ,0
Exp/Cntr=0.3,0.1

Type RM Length L Ch R = 1 ,91015   ,848,848,848
BEGIN DESCRIPTION:
MILLER CREEK 144.0
END DESCRIPTION:
XS GIS Cut Line= 4
      2910619.93     10043264.11       2911161.6     10041847.44
      2911842.16       10041778.      2912508.52     10041028.33
#Sta/Elev= 30
  3220.2 1320.94  3579.6 1309.54  3771.6  1298.3  4055.7 1284.03  4216.3 1268.33
  4260.8  1272.1  4448.4  1275.6  4571.6 1274.36  4614.9    1274  4675.3 1274.43
  4753.8 1273.77    4897 1255.03  4992.1 1245.52  4994.8 1245.02  4998.1 1245.52
  5045.4  1246.3  5095.6 1254.73  5155.9 1259.46  5231.9    1259  5260.3 1259.03
  5491.1 1269.77  5558.5  1272.2  5768.5 1275.01  5825.4 1277.94  5903.1 1287.49
  6009.3 1306.21    6052    1317    6236 1371.24  6363.3 1416.77    6424 1420.34
#Mann= 15 ,-1 , 0
  3220.2      .1       0  3579.6     .05       0  3771.6      .1       0
  4260.8     .16       0  4448.4      .1       0  4571.6     .05       0
  4614.9      .1       0  4675.3     .05       0    4897     .16       0
  4992.1     .07       0  4998.1     .16       0  5231.9      .1       0
  5260.3     .16       0  5491.1      .1       0  5558.5     .16       0
#XS Ineff= 2 , 0
         4445.74 1276.97
Permanent Ineff=
       T       T
Bank Sta=4897,5095.6
XS Rating Curve= 0 ,0
Exp/Cntr=0.3,0.1

Type RM Length L Ch R = 1 ,90167   ,736,736,736
BEGIN DESCRIPTION:
MILLER CREEK 141.0
END DESCRIPTION:
XS GIS Cut Line= 3
      2911335.22     10043875.21      2911737.99       10042653.
       2912647.7      10041229.4
#Sta/Elev= 30
  3162.5 1328.43  3769.7 1308.72  3871.8 1307.79  3973.9 1310.47  4076.1  1308.3
  4178.2 1304.16  4199.9 1303.19  4379.2 1284.97  4433.9 1271.75  4498.2  1268.1
  4732.7 1266.72    4781 1260.92  4817.4 1251.29  4884.2 1241.86  4938.8 1239.63
  4978.1 1241.01  4990.3 1237.85    4993 1237.35  4996.3 1237.85 5046.31 1252.44
    5072 1262.49  5240.1 1270.12  5520.3 1272.37    5625 1284.01  5817.2 1314.09
  5905.2 1337.14  5999.1 1355.28  6041.4  1358.8  6129.3  1385.6  6138.8 1384.86
#Mann= 14 ,-1 , 0
  3162.5      .1       0  3769.7     .05       0  3871.8      .1       0
  3973.9     .05       0  4076.1      .1       0  4178.2     .16       0
  4199.9     .05       0  4379.2     .16       0  4498.2     .05       0
  4938.8     .16       0  4990.3     .07       0  4996.3     .16       0
  5240.1      .1       0    5625     .16       0
Bank Sta=4817.4,5046.31
XS Rating Curve= 0 ,0
Exp/Cntr=0.3,0.1

Type RM Length L Ch R = 1 ,89431   ,713,713,713
BEGIN DESCRIPTION:
MILLER CREEK 140.0
END DESCRIPTION:
XS GIS Cut Line= 3
      2912293.55     10044146.02      2912633.82     10042771.05
      2912772.71     10040854.43
#Sta/Elev= 30
  3356.9 1331.65  3547.5 1323.22  3585.9 1322.07  3686.1  1317.8  3922.4 1310.92
  4187.5 1305.84  4266.4 1303.58    4410 1295.36    4544 1298.64  4830.8 1288.82
    4881 1276.24    4901 1248.58  4906.4 1242.42  4956.1  1238.3  4978.2 1237.85
    4981 1237.35  4984.2 1237.85  5111.6 1249.55  5182.1 1259.53  5883.6  1267.3
  5953.8 1276.42  5996.8  1290.3  6084.1  1312.4  6150.6 1336.52  6254.5 1360.27
    6290 1375.08  6344.8 1385.37  6424.4  1412.5  6592.1 1422.67    6695 1426.77
#Mann= 13 ,-1 , 0
  3356.9      .1       0  3547.5     .05       0  3585.9      .1       0
  3686.1     .05       0  3922.4      .1       0  4187.5     .05       0
  4266.4      .1       0  4956.1     .16       0  4978.2     .07       0
  4984.2     .16       0  5182.1     .05       0  5996.8     .16       0
  6592.1      .1       0
#XS Ineff= 1 ,-1
 5180.27 5192.29 1259.65
Permanent Ineff=
       T
Bank Sta=4901,5111.6
XS Rating Curve= 0 ,0
Exp/Cntr=0.3,0.1

Type RM Length L Ch R = 1 ,88718   ,903,903,903
BEGIN DESCRIPTION:
MILLER CREEK 139.0
END DESCRIPTION:
XS GIS Cut Line= 4
      2912675.47     10044062.75      2913307.43     10042882.16
      2913418.55     10041687.72      2913307.45     10040618.46
#Sta/Elev= 30
  3331.3 1316.42  4052.5 1290.57  4124.5 1288.71  4233.6 1285.32  4342.7 1282.14
  4451.8 1279.43  4536.3 1280.32  4560.9 1279.59  4669.9 1273.19    4709 1260.15
    4844 1258.73  4866.8 1253.69  4889.8 1245.32  4965.2 1234.79  4987.2 1233.39
  4989.9 1232.89  4993.2 1233.39  5040.4 1233.83    5162  1245.3  5166.7 1245.69
    5412 1261.11  5964.5 1259.84  6075.1 1263.05  6192.8 1274.03  6308.8 1289.78
  6402.4 1321.99  6557.7  1356.8  6728.6 1409.83  6887.8 1413.63    6945 1414.98
#Mann= 16 ,-1 , 0
  3331.3      .1       0  4052.5     .05       0  4124.5      .1       0
  4233.6     .16       0  4342.7     .05       0  4451.8      .1       0
  4536.3     .16       0  4560.9      .1       0  4669.9     .16       0
  4866.8     .05       0  4965.2     .16       0  4987.2     .07       0
  4993.2     .16       0    5162     .05       0  6192.8     .16       0
  6887.8      .1       0
Bank Sta=4889.8,5166.7
XS Rating Curve= 0 ,0
Exp/Cntr=0.3,0.1

Type RM Length L Ch R = 1 ,87815   ,556,556,556
BEGIN DESCRIPTION:
MILLER CREEK 138.0
END DESCRIPTION:
XS GIS Cut Line= 4
      2913128.59      10043566.2      2914040.07     10043050.56
      2914336.95     10042279.73      2914446.24     10041087.88
#Sta/Elev= 30
  3498.3 1288.46  3722.1 1277.77  3838.2 1274.23  3860.9 1272.85  3956.1 1272.09
  4186.7  1253.9  4246.6 1259.95  4306.8 1264.56  4442.4  1265.1  4490.1 1264.35
  4556.6 1257.32  4650.1 1255.31  4815.2    1247  4895.8 1238.06  5025.8 1233.34
  5028.6 1232.84  5031.8 1233.34  5077.9 1237.33  5105.9 1241.22  5185.1 1251.41
  5451.3  1252.9    6045 1257.96  6150.8 1263.01  6170.9  1267.8  6200.6 1269.36
  6221.1 1270.87    6299 1290.56  6331.6 1302.84  6427.7 1329.22  6568.4 1339.81
#Mann= 16 ,-1 , 0
  3498.3     .16       0  3722.1      .1       0  3838.2     .16       0
  3860.9      .1       0  4186.7     .05       0  4246.6      .1       0
  4442.4     .16       0  4650.1      .1       0  4815.2     .05       0
  5025.8     .04       0  5031.8     .05       0  5105.9      .1       0
  5451.3     .05       0    6045     .16       0  6200.6     .05       0
    6299     .16       0
Bank Sta=4895.8,5077.9
XS Rating Curve= 0 ,0
Exp/Cntr=0.3,0.1

Type RM Length L Ch R = 1 ,87259   ,411,411,411
BEGIN DESCRIPTION:
MILLER CREEK 137.0
END DESCRIPTION:
XS GIS Cut Line= 4
      2914279.66     10044842.22      2914576.53     10043212.02
      2914701.53     10042435.98      2914769.24      10041274.5
#Sta/Elev= 30
  3107.4 1286.34  3518.4 1272.55    3592 1273.19  3671.6 1268.34  4211.7 1253.33
  4454.4  1250.3    4649 1244.83  4747.4 1243.75  4803.1 1237.82  4808.1 1241.08
  4843.7  1232.8  4884.2 1224.74  4995.7 1221.56  4998.4 1221.06  5001.7 1221.56
    5050 1232.02  5066.5 1242.84  5105.2 1243.47  5142.7 1244.11    5374 1244.59
  5441.6 1248.09  5572.4 1247.11  6144.7 1256.96  6193.8 1258.14  6223.8 1265.35
    6275 1267.64  6322.7 1276.58    6421  1288.9  6654.6 1307.25  6713.9 1318.66
#Mann= 15 ,-1 , 0
  3107.4     .08       0    3592      .1       0  3671.6     .08       0
  4211.7     .05       0  4454.4     .08       0    4649     .05       0
  4995.7     .04       0  5001.7     .05       0  5105.2     .08       0
  5142.7     .05       0    5374     .08       0  5572.4     .05       0
  6144.7     .16       0  6322.7     .05       0    6421     .16       0
#XS Ineff= 1 ,-1
 4740.91 4811.36 1240.65
Permanent Ineff=
       T
Bank Sta=4843.7,5050
XS Rating Curve= 0 ,0
Exp/Cntr=0.3,0.1

Type RM Length L Ch R = 1 ,86848   ,397,397,397
BEGIN DESCRIPTION:
MILLER CREEK 136.0
END DESCRIPTION:
XS GIS Cut Line= 4
      2914545.27     10044837.06       2914805.7     10043534.94
      2914987.99     10042467.23      2915373.41     10041680.76
#Sta/Elev= 30
  3440.8 1294.07  3583.2 1285.65  3876.1  1280.6    3980 1277.77  4091.4 1273.58
  4269.8 1268.99    4413 1264.45  4525.2 1241.43    4654 1248.22  4731.1 1237.98
  4767.1 1234.51  4830.8 1230.53  4866.2 1228.52  4969.8 1221.04  4972.6 1220.54
  4975.8 1221.04  5155.4 1230.89  5262.5 1233.68  5361.5 1236.47  5460.6 1245.04
  5469.5 1244.79  6011.7  1245.9  6200.3  1250.6  6256.7 1269.75  6368.9 1275.66
  6413.9 1286.98  6540.6 1303.24  6579.6 1306.81  6616.4 1318.42  6727.7 1328.77
#Mann= 15 ,-1 , 0
  3440.8     .08       0  3876.1      .1       0    3980     .08       0
  4091.4      .1       0  4269.8     .08       0  4731.1     .05       0
  4767.1     .16       0  4866.2     .08       0  4969.8     .07       0
  4975.8     .08       0  5262.5     .05       0  5361.5      .1       0
  5460.6     .08       0  5469.5     .05       0  6540.6     .16       0
#XS Ineff= 4 ,-1
  3440.8 4654.55 1247.78 5225.44 5247.81 1232.98 5286.59 5300.31 1234.45
 5406.51 5433.65 1240.64
Permanent Ineff=
       T       T       T       T
Bank Sta=4830.8,5155.4
XS Rating Curve= 0 ,0
Exp/Cntr=0.3,0.1

Type RM Length L Ch R = 1 ,86451   ,625,625,625
BEGIN DESCRIPTION:
MILLER CREEK 135.0
END DESCRIPTION:
XS GIS Cut Line= 4
      2914644.24     10044847.45      2914899.45     10044066.19
      2915034.87     10043368.27      2915415.08     10041889.08
#Sta/Elev= 30
  3734.4 1296.97  4453.1 1275.54  4721.8 1264.07  4864.4 1231.96  4905.1 1228.23
  4947.9 1221.34  4996.6 1221.13  4999.4 1220.63  5002.6 1221.13  5061.7 1224.19
  5186.8 1224.15  5231.1 1227.13  5258.2 1234.41  5286.4 1235.15  5398.5 1243.86
  5476.4 1247.06  5509.4 1245.94    5539 1230.04  5571.3 1229.27  5701.9 1232.12
  5788.6 1247.98  5889.1  1246.2  5932.7 1241.19  6314.7 1250.37  6366.4 1246.55
  6397.3 1257.61    6449 1256.85  6525.7 1265.26  6628.5 1276.65  6794.5 1308.65
#Mann= 11 ,-1 , 0
  3734.4      .1       0  4453.1     .16       0  4996.6     .07       0
  5002.6     .16       0  5061.7      .1       0  5186.8     .05       0
  5286.4      .1       0  5398.5     .05       0  5476.4      .1       0
  5889.1     .05       0  6525.7     .16       0
#XS Ineff= 3 ,-1
  5258.2 5286.73 1234.35 5299.03 5331.47 1238.21 5502.62 5786.19 1247.21
Permanent Ineff=
       T       T       T
Bank Sta=4905.1,5231.1
XS Rating Curve= 0 ,0
Exp/Cntr=0.3,0.1

Type RM Length L Ch R = 1 ,85826   ,293,293,293
BEGIN DESCRIPTION:
MILLER CREEK 134.0
END DESCRIPTION:
XS GIS Cut Line= 3
      2915956.76     10044436.02      2915420.28     10043222.44
      2915472.37     10041800.56
#Sta/Elev= 30
  3944.8 1295.19  4121.4 1291.08  4155.7  1286.8  4272.2 1282.11  4322.6 1275.66
  4782.9  1247.9  4869.6 1238.56  4898.5 1228.32    4975 1211.89  4994.1 1211.67
  4996.8 1211.17  5000.1 1211.67  5029.7 1212.98  5106.3 1227.13  5111.8 1227.18
  5221.4 1228.49  5699.8 1243.72  5834.3 1240.68  5920.8 1237.54  6032.1 1246.07
  6080.9 1247.74  6120.9 1244.49    6151 1252.55    6191 1252.19  6235.8 1257.37
  6321.1 1264.11  6421.1  1277.2  6501.2 1292.36  6601.3 1320.71  6694.5 1329.04
#Mann= 11 ,-1 , 0
  3944.8      .1       0  4322.6     .16       0  4782.9     .05       0
  4994.1    .035       0  5000.1     .05       0  5111.8      .1       0
  5221.4     .05       0  5699.8     .16       0  5834.3     .05       0
  6032.1     .08       0  6235.8     .16       0
Bank Sta=4898.5,5106.3
XS Rating Curve= 0 ,0
Exp/Cntr=0.3,0.1

Type RM Length L Ch R = 1 ,85533   ,1104,1104,1104
BEGIN DESCRIPTION:
MILLER CREEK 133.0
END DESCRIPTION:
XS GIS Cut Line= 3
      2916210.11     10044003.23       2915550.4     10042961.59
      2915758.74       10042031.
#Sta/Elev= 30
    4223  1283.2  4480.3  1265.4  4629.3 1257.36    4681 1249.82  4738.7 1245.82
  4926.8 1243.01  4956.3 1226.55  4978.5 1214.68  4996.7 1210.64  4999.5 1210.14
  5002.7 1210.64    5077 1223.14  5093.8 1224.89  5172.5 1224.67  5196.7 1225.17
  5291.7 1226.14  5370.1 1226.92  5441.6 1231.41  5512.9 1239.99  5596.2 1241.47
  5787.3  1235.7  5894.4 1237.36  5994.5 1245.49  6058.4 1243.35  6089.1 1250.24
  6212.1 1261.11  6242.8 1266.66  6304.3 1286.43  6334.8  1291.3  6409.6 1321.53
#Mann= 12 ,-1 , 0
    4223      .1       0  4480.3     .16       0  4996.7     .07       0
  5002.7     .16       0    5077      .1       0  5172.5     .05       0
  5196.7      .1       0  5291.7     .05       0  5596.2     .16       0
  5787.3     .05       0  5994.5     .08       0  6212.1     .16       0
Bank Sta=4956.3,5093.8
XS Rating Curve= 0 ,0
Exp/Cntr=0.3,0.1

Type RM Length L Ch R = 1 ,84429   ,477,477,477
BEGIN DESCRIPTION:
MILLER CREEK 131.0
END DESCRIPTION:
XS GIS Cut Line= 3
      2916355.96     10043940.75      2916418.46     10042642.14
      2916245.28     10041977.14
#Sta/Elev= 30
    3502 1278.82    3840 1258.83  3949.5 1248.01  4066.8 1240.35  4480.2 1236.44
  4540.2 1234.67  4730.4 1222.21  4808.6 1219.23  4825.9  1219.1  4905.1 1217.61
  4965.8 1212.11  5018.5 1211.34  5021.2 1210.84  5024.5 1211.34  5038.1 1220.44
  5056.8 1231.66    5062 1227.12  5069.1 1234.68  5079.5 1237.56  5117.2  1240.3
  5162.1 1240.13  5183.5 1245.11  5224.1 1264.57  5234.8 1267.61  5265.5 1283.71
  5299.9 1294.03  5337.6 1310.99  5348.1 1315.96  5389.5 1325.51  5489.3 1340.22
#Mann= 10 ,-1 , 0
    3502      .1       0    3840     .16       0  4066.8     .05       0
  4808.6      .1       0  4825.9     .05       0  5018.5     .04       0
  5024.5     .05       0  5117.2      .1       0  5234.8     .08       0
  5337.6     .16       0
Bank Sta=4730.4,5038.1
XS Rating Curve= 0 ,0
Exp/Cntr=0.3,0.1

Type RM Length L Ch R = 1 ,83952   ,697,697,697
BEGIN DESCRIPTION:
MILLER CREEK 130.0
END DESCRIPTION:
XS GIS Cut Line= 3
      2916710.12     10043996.35      2916904.57     10043051.87
      2916557.36     10041899.12
#Sta/Elev= 30
  3597.6 1272.88  3906.6 1262.55  4141.4 1257.44  4208.5 1246.83    4315 1238.44
  4468.1 1234.77  4519.2 1235.73  4565.4    1233  4806.9 1234.99  4845.1 1233.06
  4904.4 1218.51  4949.4 1211.15    5006 1210.87  5008.8 1210.37    5012 1210.87
  5086.6 1215.35  5113.5 1219.29  5165.7  1228.7  5203.5 1230.18    5351 1235.46
  5458.1 1235.06  5515.7 1239.13  5531.2 1240.99  5562.6 1250.19  5614.8 1281.48
  5640.7 1286.55    5667 1295.64  5687.9 1306.84    5712 1315.15  5765.8 1321.44
#Mann= 7 ,-1 , 0
  3597.6     .05       0  4904.4      .1       0    5006     .07       0
    5012      .1       0  5203.5     .05       0    5351     .08       0
  5515.7     .16       0
Bank Sta=4904.4,5113.5
XS Rating Curve= 0 ,0
Exp/Cntr=0.3,0.1

Type RM Length L Ch R = 1 ,83255   ,740,740,740
BEGIN DESCRIPTION:
MILLER CREEK 129.0
END DESCRIPTION:
XS GIS Cut Line= 4
      2917293.46     10043815.74      2917411.51     10042843.53
      2917314.29     10042031.03      2916717.65     10041358.08
#Sta/Elev= 30
  3510.7 1258.89    3783 1251.26  3875.4 1243.57  3973.7 1241.06  4039.3 1238.42
  4375.1 1230.64  4556.6 1224.84  4600.6 1229.38  4726.3 1228.91  4872.6 1215.21
  4907.4 1212.93  4943.1 1211.44  4970.8 1206.85  4990.4  1200.8  4993.2  1200.3
  4996.4  1200.8  5033.7 1202.66  5060.8 1211.37  5094.1 1215.75  5130.1 1223.29
  5154.6 1229.89  5269.5 1229.74  5544.7 1233.67  5622.5  1236.2  5664.9 1241.75
  5714.5 1260.29  5947.8 1281.76  5994.3 1283.42  6068.2 1292.03  6207.7 1295.35
#Mann= 13 ,-1 , 0
  3510.7     .05       0    3783      .1       0  3973.7     .05       0
  4039.3      .1       0  4375.1     .05       0  4907.4      .1       0
  4970.8     .05       0  4990.4     .04       0  4996.4     .05       0
  5130.1     .08       0  5269.5     .05       0  5664.9     .16       0
  5994.3      .1       0
#XS Ineff= 2 , 0
         4604.55 1229.54
Permanent Ineff=
       T       T
Bank Sta=4872.6,5094.1
XS Rating Curve= 0 ,0
Exp/Cntr=0.3,0.1

Type RM Length L Ch R = 1 ,82515   ,797,797,797
BEGIN DESCRIPTION:
MILLER CREEK 128.0
END DESCRIPTION:
XS GIS Cut Line= 3
      2917428.63     10043907.44      2917735.92     10042657.44
      2918213.67     10042158.92
#Sta/Elev= 30
  3291.9 1261.02  3594.3 1247.76  3756.7 1242.66  3820.8 1240.32  3851.7 1240.89
  3913.6 1237.68  3965.1 1237.96  4006.3 1235.59  4111.2 1232.66  4140.1  1233.4
  4181.3 1230.78  4230.7 1230.98  4277.4 1227.93    4377 1226.32    4402 1222.12
  4407.9    1219  4459.4 1223.84  4568.2 1226.48  4802.9 1221.04  4880.6 1213.83
  4944.4 1208.37  4997.7 1198.51  5000.4 1198.01  5003.7 1198.51  5113.9 1211.45
  5128.1 1214.68  5156.4 1221.16  5191.9 1222.14  5220.2  1226.3  5269.6 1227.58
#Mann= 5 ,-1 , 0
  3291.9     .05       0  3756.7      .1       0  3820.8     .05       0
  4997.7    .035       0  5003.7     .05       0
#XS Ineff= 2 , 0
         4565.34 1226.75
Permanent Ineff=
       T       T
Bank Sta=4880.6,5128.1
XS Rating Curve= 0 ,0
Exp/Cntr=0.3,0.1

Type RM Length L Ch R = 1 ,81718   ,862,862,862
BEGIN DESCRIPTION:
MILLER CREEK 126.0
END DESCRIPTION:
XS GIS Cut Line= 4
      2917678.65     10043985.54      2918433.84      10043256.4
      2918558.84      10042631.4      2918315.01     10042237.12
#Sta/Elev= 30
  3542.8 1267.01  3720.8 1264.63  3989.4 1258.83  4109.8 1257.95    4329 1252.19
  4420.8 1247.98  4596.5 1245.42  4748.5 1238.13  4777.9  1235.7  4811.3 1232.84
  4880.8 1226.45  4896.3  1223.1  4901.4  1223.9    4942 1215.61  4947.3 1211.45
  4962.4  1205.7  4972.6 1199.38  5000.4 1195.63  5003.2 1195.13  5006.4 1195.63
  5013.4 1195.75  5033.8 1201.61  5064.4 1205.55  5166.4 1211.73  5235.9 1216.91
  5279.1 1218.36  5294.5 1220.37  5358.3 1220.92  5510.8 1225.46  5693.5 1225.54
#Mann= 6 ,-1 , 0
  3542.8      .1       0  4777.9     .16       0  4811.3      .1       0
  5000.4     .07       0  5006.4      .1       0  5235.9     .05       0
Bank Sta=4947.3,5166.4
XS Rating Curve= 0 ,0
Exp/Cntr=0.3,0.1

Type RM Length L Ch R = 1 ,80856   ,1053,1053,1053
BEGIN DESCRIPTION:
MILLER CREEK 124.0
END DESCRIPTION:
XS GIS Cut Line= 3
      2917675.38     10044093.55      2919029.57     10043239.37
      2920369.83     10042190.77
#Sta/Elev= 30
  3067.6 1271.01  3980.2 1254.36  4176.8 1248.07  4219.9 1247.92  4540.9 1242.52
  4635.1 1235.89  4665.1 1229.42  4686.1 1229.85  4701.9 1223.96  4885.1 1207.52
    4914 1205.86    4996 1190.79  4998.8 1190.29    5002 1190.79  5090.7 1204.24
  5135.5 1207.88    5146 1209.32  5213.2 1215.64  5314.5 1211.61    5391 1207.67
  5419.5 1199.99  5462.9 1204.97  5558.2 1207.23  6011.7 1217.89  6067.8 1220.37
  6120.8 1228.98  6210.7  1268.3  6274.9 1285.68  6310.2 1289.31  6370.4 1302.72
#Mann= 12 ,-1 , 0
  3067.6      .1       0  3980.2     .16       0  4176.8      .1       0
  4219.9     .16       0  4701.9      .1       0    4996     .07       0
    5002      .1       0  5090.7     .16       0    5146     .05       0
  5314.5      .1       0  5558.2     .05       0  6120.8     .16       0
#XS Ineff= 2 , 0
                         5211.36         1215.92
Permanent Ineff=
       T       T
Bank Sta=4885.1,5135.5
XS Rating Curve= 0 ,0
Exp/Cntr=0.3,0.1

Type RM Length L Ch R = 1 ,79803   ,674,674,674
BEGIN DESCRIPTION:
MILLER CREEK 123.0
END DESCRIPTION:
XS GIS Cut Line= 4
      2917689.08     10044178.25      2918293.21     10043777.23
      2919058.84     10043782.44      2919678.61      10043115.8
#Sta/Elev= 30
  3792.5 1273.75  4062.3 1270.59  4555.2 1258.62  4648.8 1254.48  4712.9 1253.25
  4738.2 1250.04  4827.4 1245.69  4922.9 1239.86  4942.9 1232.46  4960.2 1219.95
  4972.9 1201.95  4982.9 1188.35  4999.9 1184.31  5002.6 1183.81  5005.9 1184.31
  5022.9 1191.99  5042.9 1191.05  5072.9 1196.16  5122.9 1198.07  5162.9 1202.42
  5232.9 1208.63  5325.1 1211.45  5330.3 1211.28    5627 1214.97  5697.1 1214.35
  5756.2 1213.82  6000.8  1215.6  6014.6  1215.7  6152.7 1214.96  6193.5  1214.2
#Mann= 15 ,-1 , 0
  3792.5      .1       0  4555.2     .16       0  4648.8      .1       0
  4827.4     .16       0  4960.2      .1       0  4999.9     .07       0
  5005.9      .1       0  5325.1     .16       0  5330.3      .1       0
    5627     .05       0  5697.1      .1       0  5756.2     .05       0
  6000.8      .1       0  6014.6     .05       0  6152.7      .1       0
#XS Ineff= 2 , 0
                         5557.39         1214.61
Permanent Ineff=
       T       T
Bank Sta=4972.9,5162.9
XS Rating Curve= 0 ,0
Exp/Cntr=0.3,0.1

Type RM Length L Ch R = 1 ,79129   ,898,898,898
BEGIN DESCRIPTION:
MILLER CREEK 121.0
END DESCRIPTION:
XS GIS Cut Line= 4
      2917970.33     10044855.34      2918881.76      10044568.9
      2919511.96     10043855.35      2919730.33     10043127.48
#Sta/Elev= 30
  3706.2  1283.5  3756.5 1278.95  3955.8 1275.69  4026.2 1269.56  4217.9    1269
  4532.8 1258.06  4689.7 1253.91  4773.2 1251.15  4834.7 1246.86  4918.1 1233.09
  4932.4 1226.02  4946.6 1215.03  4960.8 1199.77    4975 1186.24  4992.9 1181.25
  4995.7 1180.75  4998.9 1181.25  5005.9 1182.21    5031 1192.23    5048 1194.21
  5095.4 1198.69  5394.4 1208.48  5477.8 1212.15    5626 1211.38  5938.7 1212.98
  6040.1 1213.34  6054.1 1213.44  6141.5 1212.88  6344.3 1213.36  6373.5 1213.45
#Mann= 16 ,-1 , 0
  3706.2      .1       0  4532.8     .05       0  4689.7      .1       0
  4773.2     .05       0  4834.7      .1       0  4992.9     .07       0
  4998.9      .1       0  5005.9     .16       0    5048     .05       0
  5394.4      .1       0    5626     .05       0  5938.7      .1       0
  6040.1     .05       0  6054.1      .1       0  6141.5     .05       0
  6344.3      .1       0
Bank Sta=4960.8,5095.4
XS Rating Curve= 0 ,0
Exp/Cntr=0.3,0.1

Type RM Length L Ch R = 1 ,78231   ,946,946,946
BEGIN DESCRIPTION:
MILLER CREEK 120.0
END DESCRIPTION:
XS GIS Cut Line= 4
      2919709.87     10045391.84      2919954.67     10044907.44
      2919949.46      10044011.6       2919783.4     10043119.02
#Sta/Elev= 30
    3984 1258.19  4109.4 1254.48  4418.9  1243.1  4729.1 1241.18  4760.1 1239.91
  4860.5 1233.66  4870.5 1229.75  4880.5 1219.26  4890.5 1199.96 4897.73 1193.92
  4900.5 1190.21  4923.7 1187.26  4997.5  1179.2  5000.2  1178.7  5003.5  1179.2
  5020.5 1182.67  5040.5 1193.84  5120.5 1202.79  5291.2    1206  5355.1 1206.38
  5654.4 1208.45  5671.9 1206.54  5676.9 1208.54  5724.6 1205.44  5729.7 1207.95
  5756.1 1208.69  5918.8 1204.01  6189.6 1209.35  6290.5 1211.61  6330.5 1212.95
#Mann= 11 ,-1 , 0
    3984      .1       0  4109.4     .16       0  4729.1      .1       0
  4760.1     .16       0  4923.7     .05       0  4997.5    .035       0
  5003.5     .05       0  5291.2     .16       0  5355.1     .05       0
  6189.6      .1       0  6290.5     .05       0
#XS Ineff= 2 , 0
                         5507.95         1207.68
Permanent Ineff=
       T       T
Bank Sta=4897.73,5040.5
XS Rating Curve= 0 ,0
Exp/Cntr=0.3,0.1

Type RM Length L Ch R = 1 ,77285   ,506,506,506
BEGIN DESCRIPTION:
MILLER CREEK 118.0
END DESCRIPTION:
XS GIS Cut Line= 4
       2920362.9     10045031.04       2920800.4      10044447.7
      2920793.46     10043586.59      2920661.51     10042961.58
#Sta/Elev= 30
  3892.4 1227.05    4048 1221.71    4071 1221.25  4344.1 1218.76  4409.7 1219.49
  4582.4 1215.03  4584.1 1214.92  4687.6 1208.45  4815.5 1201.46  4875.5 1190.43
  4915.5 1183.85  4965.6 1183.01  4992.6 1177.67  4995.3 1177.17  4998.6 1177.67
  5035.6  1179.1  5085.6 1190.14  5133.4 1196.76    5278 1199.94  5376.4 1201.54
  5513.9 1202.53    5576 1204.35  5618.5  1207.7  5677.5 1217.44  5761.6  1226.7
  5963.8 1295.68  5996.7 1303.77  6047.8 1311.16  6063.4 1316.47  6121.5 1320.03
#Mann= 16 ,-1 , 0
  3892.4     .16       0    4048      .1       0    4071     .16       0
  4344.1      .1       0  4409.7     .05       0  4582.4      .1       0
  4584.1     .05       0  4687.6      .1       0  4992.6     .07       0
  4998.6      .1       0  5133.4     .05       0    5278      .1       0
  5376.4     .05       0  5513.9      .1       0    5576     .05       0
  5677.5     .16       0
#XS Ineff= 2 , 0
                         5252.27          1201.9
Permanent Ineff=
       T       T
Bank Sta=4875.5,5085.6
XS Rating Curve= 0 ,0
Exp/Cntr=0.3,0.1

Type RM Length L Ch R = 1 ,76779   ,482,482,482
BEGIN DESCRIPTION:
MILLER CREEK 117.0
END DESCRIPTION:
XS GIS Cut Line= 4
      2920640.66     10044906.05      2921328.18     10044225.48
      2921258.74     10043781.03       2920960.7     10042886.94
#Sta/Elev= 30
  3792.9 1216.12  4153.6 1209.99  4286.7 1211.54    4357 1213.29  4689.3 1204.69
  4778.2 1200.47  4856.9 1197.04    4879 1192.77  4903.8 1185.19  4919.7 1181.09
  4979.2 1176.29    5002 1175.91  5004.7 1175.41    5008 1175.91  5079.4 1185.76
    5086 1187.19  5136.6 1196.37  5189.7 1197.81  5239.4 1199.16  5692.2 1198.61
    5787 1202.41  5827.1 1207.32  5920.7 1227.59  5983.9 1253.78  5989.2 1253.78
  6015.5 1267.97  6020.8 1267.35  6047.1 1281.86  6092.7 1300.29  6152.6  1314.2
#Mann= 13 ,-1 , 0
  3792.9      .1       0  4286.7     .05       0    4357      .1       0
  4689.3     .16       0  4778.2      .1       0    4879     .05       0
  4979.2      .1       0    5002     .07       0    5008      .1       0
  5079.4     .05       0  5189.7      .1       0  5239.4     .05       0
  5827.1     .16       0
Bank Sta=4903.8,5086
XS Rating Curve= 0 ,0
Exp/Cntr=0.3,0.1

Type RM Length L Ch R = 1 ,76297   ,801,801,801
BEGIN DESCRIPTION:
MILLER CREEK 116.0
END DESCRIPTION:
XS GIS Cut Line= 4
      2921432.33     10045593.58      2921842.07      10044635.2
      2921682.35     10043524.09      2921363.69     10042658.18
#Sta/Elev= 30
  3334.3 1240.27  3519.9 1230.83  4071.3 1218.04  4229.4 1209.69  4539.7 1204.33
  4576.3 1199.54  4581.4  1201.5    4661 1183.29    4762 1177.75  4832.7 1179.61
  4889.2 1177.76  4996.3 1174.06  4999.1 1173.56  5002.3 1174.06  5075.2 1180.06
  5115.6 1195.49  5189.2 1196.45  5289.2 1196.39  5376.5 1197.12  6036.1 1199.89
  6077.6 1202.23  6096.2 1207.22  6133.2 1223.08  6138.8  1229.2  6170.8  1249.5
  6194.1 1261.36  6224.6 1273.49  6256.1 1282.19  6310.7 1285.12  6421.8  1284.5
#Mann= 9 ,-1 , 0
  3334.3      .1       0  4071.3     .05       0  4889.2      .1       0
  4996.3     .07       0  5002.3      .1       0  5189.2     .05       0
  5289.2      .1       0  5376.5     .05       0  6036.1     .16       0
#XS Ineff= 2 , 0
          4801.7  1180.5
Permanent Ineff=
       T       T
Bank Sta=4832.7,5075.2
XS Rating Curve= 0 ,0
Exp/Cntr=0.3,0.1

Type RM Length L Ch R = 1 ,75496   ,430,430,430
BEGIN DESCRIPTION:
MILLER CREEK 115.0
END DESCRIPTION:
XS GIS Cut Line= 4
        2922224.     10045447.74      2922460.13     10044482.42
      2922543.46     10043489.37      2922279.58     10042531.06
#Sta/Elev= 30
  3655.1 1228.49  3875.4 1220.73  4241.5 1220.28  4400.5 1212.33  4441.6 1205.81
  4622.9 1192.46  4637.7 1191.65  4829.4 1181.78  4888.4 1171.46  4908.5 1161.76
  4995.8 1151.78  4998.5 1151.28  5001.8 1151.78  5018.9 1152.07  5045.8 1161.88
  5099.1 1171.38  5170.9 1177.24  5269.2 1186.13  5367.6 1189.99  5585.9 1191.36
  5792.6 1191.89  5993.4 1194.35    6049 1194.24  6287.5 1197.33  6418.8 1204.25
    6475 1217.13  6509.4 1243.68  6514.5 1241.81  6538.6 1251.93  6639.4 1251.52
#Mann= 14 ,-1 , 0
  3655.1      .1       0  4622.9     .16       0  4637.7      .1       0
  4829.4     .16       0  4995.8     .07       0  5001.8     .16       0
  5170.9     .05       0  5269.2      .1       0  5367.6     .05       0
  5585.9      .1       0  5792.6     .05       0  5993.4      .1       0
    6049     .05       0  6538.6      .1       0
Bank Sta=4888.4,5099.1
XS Rating Curve= 0 ,0
Exp/Cntr=0.3,0.1

Type RM Length L Ch R = 1 ,75066   ,571,571,571
BEGIN DESCRIPTION:
MILLER CREEK 114.0
END DESCRIPTION:
XS GIS Cut Line= 4
       2922876.8     10045385.15       2922925.4     10044531.03
      2922904.57      10043697.7      2922932.35     10042774.11
#Sta/Elev= 30
  3765.3 1229.09  4217.4 1210.94  4337.6 1200.47  4688.1 1188.22  4826.7 1175.53
  4898.2 1169.15  4908.2 1166.24  4918.2 1159.73  4985.2 1151.12    4988 1150.62
  4991.2 1151.12  5018.2  1151.9  5048.2 1156.17  5068.2 1162.78  5078.2 1168.41
  5095.8 1174.53  5100.9 1173.61  5172.4 1186.13  5238.3 1187.71  5270.9 1186.08
  5298.3 1188.08  5369.4 1187.62  5959.3 1188.68  6068.6 1190.99  6155.8 1198.96
  6178.7 1205.24  6228.7 1228.28  6308.7 1255.15  6334.6 1257.41  6378.4 1253.73
#Mann= 10 ,-1 , 0
  3765.3      .1       0  4826.7     .16       0  4985.2     .07       0
  4991.2     .16       0  5172.4     .05       0  5270.9      .1       0
  5369.4     .05       0  5959.3     .16       0  6155.8     .05       0
  6334.6      .1       0
Bank Sta=4908.2,5078.2
XS Rating Curve= 0 ,0
Exp/Cntr=0.3,0.1

Type RM Length L Ch R = 1 ,74495   ,610,610,610
BEGIN DESCRIPTION:
MILLER CREEK 113.0
END DESCRIPTION:
XS GIS Cut Line= 4
      2923071.22     10045447.73      2923529.57     10044531.03
      2923418.46     10043683.81      2923362.91     10042968.64
#Sta/Elev= 30
  3561.5 1227.11  3764.7 1217.33  4150.4 1191.48  4515.2 1182.59  4724.9 1183.75
  4819.7 1175.88  4862.5 1165.78  4906.4 1161.25  4956.8 1151.42  4994.2 1148.66
  4996.9 1148.16  5000.2 1148.66  5057.7 1154.37  5077.9 1163.74  5109.4 1169.75
    5119 1169.82  5167.6  1172.3  5188.8 1179.09  5246.4 1173.03  5325.2 1180.17
    5404 1179.49  5438.4    1185  5505.8 1182.54  5660.1 1187.32  5765.3 1193.88
  5832.1 1208.44  5962.5 1225.28  6019.8 1237.27  6111.4 1244.64  6158.2  1250.3
#Mann= 9 ,-1 , 0
  3561.5      .1       0  4515.2     .16       0  4819.7      .1       0
  4994.2     .07       0  5000.2      .1       0  5109.4     .16       0
    5119     .05       0  5660.1     .16       0  6111.4     .05       0
#XS Ineff= 2 , 0
                         5194.32          1179.2
Permanent Ineff=
       T       T
Bank Sta=4906.4,5077.9
XS Rating Curve= 0 ,0
Exp/Cntr=0.3,0.1

Type RM Length L Ch R = 1 ,73885   ,712,712,712
BEGIN DESCRIPTION:
MILLER CREEK 112.0
END DESCRIPTION:
XS GIS Cut Line= 4
      2923169.16     10045481.42      2923603.18     10044439.78
       2924176.1     10044240.13      2923516.36     10042990.09
#Sta/Elev= 30
  3044.8 1223.29  3234.9    1216  3293.4  1207.5  3736.5 1185.85    3996    1182
  4003.5 1182.06  4213.5 1183.97  4396.6 1182.15  4540.7 1179.22  4764.8 1179.02
  4797.9  1179.2  4833.2 1178.76  4900.3 1163.18  4945.5 1159.25  4954.1 1150.49
  4995.1 1145.55  4997.8 1145.05  5001.1 1145.55  5064.2 1147.75  5115.1  1158.3
  5132.9 1163.11  5168.6 1173.35  5246.7 1181.79    5641 1193.62  5824.4 1200.89
  5929.3 1210.75  6032.4  1222.7  6098.8 1236.55  6156.9 1240.08  6193.4 1243.44
#Mann= 16 ,-1 , 0
  3044.8      .1       0    3996     .05       0  4003.5     .16       0
  4213.5      .1       0  4396.6     .16       0  4540.7      .1       0
  4764.8     .16       0  4797.9      .1       0  4995.1     .07       0
  5001.1      .1       0  5132.9     .05       0  5246.7      .1       0
    5641     .05       0  5824.4      .1       0  5929.3     .16       0
  6156.9     .05       0
Bank Sta=4945.5,5115.1
XS Rating Curve= 0 ,0
Exp/Cntr=0.3,0.1

Type RM Length L Ch R = 1 ,73173   ,253,253,253
BEGIN DESCRIPTION:
MILLER CREEK 111.0
END DESCRIPTION:
XS GIS Cut Line= 5
       2924959.2     10045477.71      2924875.87     10044285.04
      2924782.12     10044102.75      2924506.07     10043441.29
      2923573.81     10042904.85
#Sta/Elev= 30
  3554.5 1236.94  3859.2 1230.88  3960.2 1222.46  4281.5 1214.78  4354.8 1212.36
  4420.6 1199.14  4701.3 1187.49  4822.8 1157.99    4845 1145.24  4897.7 1150.08
  4970.9  1143.7  4973.6  1143.2  4976.9  1143.7  5099.3 1149.34    5149  1155.9
  5192.5 1163.98  5328.7 1173.51  5716.8 1180.53  5815.6 1183.46  5835.9 1183.33
  6042.9 1189.83  6063.3 1190.22    6154 1193.93  6265.1 1199.26  6276.2 1199.89
  6335.5 1204.04  6400.2 1218.95  6487.3 1231.04  6489.2 1231.32  6747.4 1249.81
#Mann= 18 ,-1 , 0
  3554.5      .1       0  3960.2     .05       0  4281.5      .1       0
  4970.9     .07       0  4976.9      .1       0  5099.3     .16       0
  5192.5      .1       0  5328.7     .05       0  5716.8      .1       0
  5815.6     .05       0  5835.9      .1       0  6042.9     .05       0
  6063.3      .1       0    6154     .05       0  6265.1      .1       0
  6276.2     .05       0  6487.3     .16       0  6489.2     .05       0
#XS Ineff= 2 , 0
                         5188.35         1164.48
Permanent Ineff=
       T       T
Bank Sta=4822.8,5149
XS Rating Curve= 0 ,0
Exp/Cntr=0.3,0.1

Type RM Length L Ch R = 1 ,72920   ,494,494,494
BEGIN DESCRIPTION:
MILLER CREEK 110.0
END DESCRIPTION:
XS GIS Cut Line= 4
       2925925.4     10045204.65      2925349.01     10044586.59
      2924647.63     10043406.03      2923654.57     10042850.48
#Sta/Elev= 30
  3481.2 1246.34  3828.8 1232.08  4144.7 1227.03  4279.1 1217.43  4468.8 1211.16
  4562.3 1196.81  4809.7 1187.36  4840.9 1181.63  4876.3 1164.74  4926.6 1155.18
  4942.2 1145.24  4954.8 1143.18  4957.5 1142.68  4960.8 1143.18  5161.8 1150.56
  5181.8 1155.01    5213 1160.54  5339.5 1165.42  5396.5 1166.51  5513.9 1173.44
  6004.2 1185.85  6008.8 1185.92    6225 1192.75  6397.5 1200.47  6444.9 1206.97
  6493.8 1216.62  6553.2  1222.2  6603.8 1234.79    6664 1238.11  6837.4 1247.24
#Mann= 13 ,-1 , 0
  3481.2     .16       0  3828.8      .1       0  4954.8     .07       0
  4960.8      .1       0  5161.8     .16       0  5339.5      .1       0
  5396.5     .16       0  5513.9     .05       0  6004.2      .1       0
  6008.8     .05       0    6225      .1       0  6444.9     .16       0
    6664     .05       0
Bank Sta=4926.6,5181.8
XS Rating Curve= 0 ,0
Exp/Cntr=0.3,0.1
