HEC-RAS study MILLER CREEK.prj: MILLER CREEK Base Level Engineering

--- MILLER CREEK.g01 (geometry) --- (continued)

Type RM Length L Ch R = 1 ,72426   ,754,754,754
BEGIN DESCRIPTION:
MILLER CREEK 109.0
END DESCRIPTION:
XS GIS Cut Line= 4
      2926092.09     10044538.02      2925689.29     10043864.37
      2924585.13     10043162.98      2923883.76     10042815.77
#Sta/Elev= 30
    3749 1236.92  4036.6 1231.27  4088.1 1230.52  4137.4 1226.01  4256.9  1215.9
  4367.8 1210.85  4502.9 1198.13  4709.5 1187.33  4754.7 1180.78  4795.5 1167.05
  4918.6 1153.07  4925.8 1146.04  4936.8 1143.09  4939.6 1142.59  4942.8 1143.09
  5064.3 1144.14  5137.2 1153.22  5194.8 1156.29  5367.5 1152.11  5443.8 1157.63
  5482.7 1160.31  5513.2 1167.08  5643.7 1176.88  6139.3 1192.44  6251.1 1197.72
  6275.5 1201.89  6352.3 1216.47  6468.5 1223.83  6531.7 1234.63  6624.6 1238.44
#Mann= 11 ,-1 , 0
    3749      .1       0  4036.6     .05       0  4088.1      .1       0
  4137.4     .05       0  4502.9      .1       0  4754.7     .16       0
  4936.8     .07       0  4942.8     .16       0  5443.8     .05       0
  6275.5     .16       0  6468.5     .05       0
#XS Ineff= 2 , 0
                         5196.31         1156.27
Permanent Ineff=
       T       T
Bank Sta=4918.6,5137.2
XS Rating Curve= 0 ,0
Exp/Cntr=0.3,0.1

Type RM Length L Ch R = 1 ,71672   ,469,469,469
BEGIN DESCRIPTION:
MILLER CREEK 108.0
END DESCRIPTION:
XS GIS Cut Line= 4
      2926064.28     10043996.28      2925758.74     10043176.87
      2925022.63      10042510.2      2924432.91     10042003.74
#Sta/Elev= 30
  3739.7 1220.77  3915.3 1209.72  4252.5 1188.04  4374.6 1182.15  4454.9 1166.42
  4611.4 1157.22  4686.1 1155.07  4732.5  1155.2  4807.7 1158.38  4829.3 1153.11
  4878.6 1143.65  4953.4 1143.06  4956.1 1142.56  4959.4 1143.06  5168.6  1143.4
  5204.4 1153.24  5225.3 1159.51    5247 1158.76  5267.9 1164.34  5314.4 1168.33
  5476.6 1175.34    5880 1194.88  5919.6 1205.64  5948.8 1207.58  5990.9 1207.55
  6011.8 1220.34  6033.7 1228.04  6107.6 1236.62  6256.4 1264.05  6384.7 1274.68
#Mann= 14 ,-1 , 0
  3739.7      .1       0  3915.3     .05       0  4252.5      .1       0
  4611.4     .05       0  4686.1      .1       0  4732.5     .05       0
  4953.4    .033       0  4959.4     .05       0  5314.4      .1       0
  5476.6     .05       0    5880     .08       0  5948.8      .1       0
  6107.6     .05       0  6256.4      .1       0
#XS Ineff= 2 , 0
         4805.68 1158.75
Permanent Ineff=
       T       T
Bank Sta=4829.3,5204.4
XS Rating Curve= 0 ,0
Exp/Cntr=0.3,0.1

Type RM Length L Ch R = 1 ,71203   ,833,833,833
BEGIN DESCRIPTION:
MILLER CREEK 107.0
END DESCRIPTION:
XS GIS Cut Line= 4
      2926460.15     10043621.34      2925960.13     10042961.59
      2925557.35     10041954.64      2925286.52      10041149.1
#Sta/Elev= 30
  3794.2 1218.84  4250.7 1206.48  4330.7 1193.09  4382.1 1189.08    4465 1180.86
  4556.6 1154.63  4662.2 1151.78    4751 1155.33  4813.6 1152.52  4873.5 1147.93
  5004.5 1143.41  5007.2 1142.91  5010.5 1143.41  5136.7 1144.62  5152.2 1146.23
    5169    1153  5176.4 1156.58  5206.1 1158.32  5230.3 1164.25  5311.2 1167.62
  5627.9 1177.47  5739.2  1180.8    5787  1185.4  5944.3 1189.11  6033.1 1193.45
    6235 1207.89  6298.3  1225.7  6372.2 1240.55  6414.4 1253.89  6556.4 1277.58
#Mann= 11 ,-1 , 0
  3794.2      .1       0  4330.7     .05       0  4382.1      .1       0
  4873.5     .05       0  5004.5    .033       0  5010.5     .05       0
  5311.2     .16       0  5627.9     .05       0    5787     .08       0
  5944.3     .05       0  6033.1     .16       0
#XS Ineff= 2 , 0
         4740.91 1155.42
Permanent Ineff=
       T       T
Bank Sta=4813.6,5169
XS Rating Curve= 0 ,0
Exp/Cntr=0.3,0.1

Type RM Length L Ch R = 1 ,70370   ,476,476,476
BEGIN DESCRIPTION:
MILLER CREEK 105.0
END DESCRIPTION:
XS GIS Cut Line= 4
      2926821.23     10043350.44      2926751.79     10042753.26
      2926355.96     10041683.81       2925890.7     10041072.73
#Sta/Elev= 30
  4001.2 1216.89  4055.1 1217.02  4249.6 1214.91  4535.9 1207.03  4604.8 1204.09
  4670.4 1192.32  4743.7 1188.24  4783.2  1173.6  4854.7 1152.61  4868.5 1146.72
  4899.2 1143.88  5089.5 1143.49  5092.3 1142.99  5095.5 1143.49  5124.4 1151.91
  5178.4 1153.02  5209.7 1161.38  5334.9 1159.72    5548  1162.5  5681.6 1168.27
  5847.8 1173.05  6010.4 1182.15  6061.9 1180.88  6076.5 1185.92  6181.1 1192.33
  6211.6 1196.59  6245.4 1205.17  6340.5 1229.97  6440.3 1244.16  6510.8 1261.17
#Mann= 13 ,-1 , 0
  4001.2     .16       0  4055.1      .1       0  4535.9     .05       0
  4670.4      .1       0  4899.2     .05       0  5089.5    .033       0
  5095.5     .05       0  5334.9      .1       0    5548     .16       0
  5681.6     .05       0  6010.4     .08       0  6181.1     .05       0
  6245.4     .16       0
#XS Ineff= 2 , 0
                         5215.34          1161.9
Permanent Ineff=
       T       T
Bank Sta=4854.7,5124.4
XS Rating Curve= 0 ,0
Exp/Cntr=0.3,0.1

Type RM Length L Ch R = 1 ,69894   ,269,269,269
BEGIN DESCRIPTION:
Mapping XS 1d31ea20
END DESCRIPTION:
XS GIS Cut Line= 3
      2927101.56     10043230.38      2927110.24     10042271.15
      2926207.79     10040978.22
#Sta/Elev= 30
  3840.5 1208.37  4191.8  1203.5  4290.2 1199.36  4407.2 1195.64  4467.2  1188.7
    4557 1188.26  4799.8 1181.14  4813.3 1180.16  4837.1 1170.52  4857.6 1160.87
 4865.34 1150.51  4878.7 1143.65  4900.8 1143.62  5048.4 1143.42  5051.2 1142.92
  5054.4 1143.42  5158.7 1150.26    5162 1150.27  5194.5 1147.29  5223.5 1151.74
  5271.7 1152.15  5516.4 1159.17  5958.9 1179.99  6004.9 1178.98  6028.3 1185.87
  6136.7 1201.05  6137.1 1201.18  6171.5 1211.92  6257.8 1229.48  6376.5 1248.08
#Mann= 13 ,-1 , 0
  3840.5      .1       0  4191.8     .05       0  4290.2      .1       0
    4557     .05       0  4837.1     .16       0  4900.8     .05       0
  5048.4    .033       0  5054.4     .05       0    5162      .1       0
  5271.7     .05       0  5958.9     .08       0  6136.7     .05       0
  6137.1     .16       0
Bank Sta=4865.34,5158.7
XS Rating Curve= 0 ,0
Exp/Cntr=0.3,0.1

Type RM Length L Ch R = 1 ,69625   ,54,54,54
BEGIN DESCRIPTION:
Mapping XS bec2a497
END DESCRIPTION:
XS GIS Cut Line= 3
      2927227.43     10043169.58      2927231.77      10042093.2
      2926347.14     10041017.78
#Sta/Elev= 30
  3838.1 1203.69  4073.9    1202  4239.6 1195.44  4314.3 1192.05  4353.9 1188.34
  4450.2 1187.36    4734 1178.82    4814 1170.28    4884 1156.76    4894 1154.07
 4906.25 1146.88  4911.7 1143.15    4928 1143.62  4971.3 1144.17  5048.6 1141.83
  5051.4 1141.33  5054.6 1141.83    5108 1145.69  5144.2 1144.16  5172.6 1146.47
  5228.8 1147.26  5304.6 1150.94  5989.7 1178.81  6031.6 1177.54  6060.3 1185.09
  6152.5 1197.08  6202.4 1211.85  6228.5 1215.37  6280.6  1228.7    6307 1232.73
#Mann= 13 ,-1 , 0
  3838.1      .1       0  4239.6     .05       0  4314.3      .1       0
  4450.2     .05       0    4928      .1       0  4971.3     .05       0
  5048.6    .033       0  5054.6     .05       0  5172.6      .1       0
  5304.6     .05       0  5989.7     .08       0  6152.5     .05       0
  6228.5     .16       0
Bank Sta=4906.25,5228.8
XS Rating Curve= 0 ,0
Exp/Cntr=0.3,0.1

Type RM Length L Ch R = 1 ,69571   ,144,144,144
BEGIN DESCRIPTION:
MILLER CREEK 104.0
END DESCRIPTION:
XS GIS Cut Line= 3
      2927275.17     10043148.77      2927282.12     10042086.26
      2926486.99     10041023.77
#Sta/Elev= 30
  3847.4 1202.57  4052.4 1201.44  4239.5  1193.4  4250.2  1193.3  4421.2 1186.99
  4712.5 1178.16  4752.5 1170.57  4792.5 1169.32  4862.5 1155.58  4921.9 1137.99
  4937.8 1135.17  4968.9 1126.04  4971.6 1125.54  4974.9 1126.04  5028.1 1126.99
  5048.9 1131.97  5078.1 1138.86  5186.5 1146.03  5204.7 1144.91  5273.3  1149.4
  5407.4 1156.15    5943 1176.87  5963.8    1175  5996.6 1177.74    6043  1176.3
  6063.9 1184.58  6143.1  1194.6  6161.6  1198.9  6199.6 1210.69    6237 1216.01
#Mann= 12 ,-1 , 0
  3847.4      .1       0  4239.5     .05       0  4250.2      .1       0
  4421.2     .05       0  4937.8      .1       0  4968.9     .07       0
  4974.9      .1       0  5048.9     .05       0  5204.7      .1       0
  5273.3     .05       0  5996.6     .08       0  6161.6     .05       0
Bank Sta=4921.9,5078.1
XS Rating Curve= 0 ,0
Exp/Cntr=0.3,0.1

Type RM Length L Ch R = 1 ,69427   ,884,884,884
BEGIN DESCRIPTION:
Mapping XS 8a1f8864
END DESCRIPTION:
XS GIS Cut Line= 4
      2927632.81     10042585.39      2927654.51     10042116.64
      2927302.95      10041908.3      2926561.76     10040937.39
#Sta/Elev= 30
  4156.1 1183.23  4233.4 1181.19    4378 1177.94  4429.9 1173.08  4627.7 1161.61
  4719.4 1160.22  4777.9 1154.94  4799.4 1157.03  4836.4 1149.46  4857.8  1148.9
  4894.9  1137.7  4925.1 1130.55  5001.3 1124.59  5004.1 1124.09  5007.3 1124.59
  5039.8 1125.03  5068.7 1127.01  5097.7 1135.52  5118.5 1137.93  5167.7 1144.26
  5278.5 1148.43  5889.5 1175.69  5924.9 1176.63  5939.4 1173.52    6003 1176.26
  6024.7  1174.7  6046.2 1184.09    6116 1193.64  6190.9 1212.55  6255.5 1225.96
#Mann= 13 ,-1 , 0
  4156.1      .1       0  4233.4     .05       0  4429.9      .1       0
  4627.7     .05       0  4925.1      .1       0  5001.3     .07       0
  5007.3      .1       0  5039.8     .05       0  5167.7      .1       0
  5278.5     .05       0    6003     .08       0    6116     .05       0
  6190.9     .16       0
Bank Sta=4894.9,5118.5
XS Rating Curve= 0 ,0
Exp/Cntr=0.3,0.1

Type RM Length L Ch R = 1 ,68543   ,405,405,405
BEGIN DESCRIPTION:
MILLER CREEK 102.0
END DESCRIPTION:
XS GIS Cut Line= 3
      2927669.77     10042585.26      2928023.93      10041408.2
      2927222.63     10040461.21
#Sta/Elev= 30
  3581.1 1182.99  3659.1 1180.96  3781.1 1178.32  3861.9 1171.23  3980.2  1160.7
  4053.6 1157.85  4166.2 1155.71  4364.3 1155.54  4369.1 1155.71  4633.7 1156.04
  4814.4 1148.49  4845.4 1147.32  4888.3 1135.53  4902.6 1129.62  4991.9 1123.26
  4994.6 1122.76  4997.9 1123.26  5030.8  1126.3  5072.9 1135.56    5108 1143.01
  5214.6 1151.08  5384.1 1152.72  5612.3  1155.6  5676.1 1161.05  5728.9 1161.47
  5793.8 1161.81  5881.5 1174.54  5966.4 1201.77  5982.2  1207.4  6050.8 1212.23
#Mann= 16 ,-1 , 0
  3581.1      .1       0  3659.1     .05       0  3861.9      .1       0
  4053.6     .16       0  4166.2      .1       0  4364.3     .16       0
  4369.1      .1       0  4814.4     .05       0  4991.9     .04       0
  4997.9     .05       0  5030.8      .1       0  5384.1     .05       0
  5728.9     .08       0  5793.8     .05       0  5966.4     .16       0
  5982.2     .05       0
#XS Ineff= 1 ,-1
 5130.27 5155.72 1144.31
Permanent Ineff=
       T
Bank Sta=4888.3,5072.9
XS Rating Curve= 0 ,0
Exp/Cntr=0.3,0.1

Type RM Length L Ch R = 1 ,68138   ,831,831,831
BEGIN DESCRIPTION:
MILLER CREEK 101.0
END DESCRIPTION:
XS GIS Cut Line= 4
      2927742.67     10042616.56      2928174.97     10041632.16
      2928305.18     10040585.29      2929008.29     10039340.52
#Sta/Elev= 30
  3361.6 1182.19  3441.6 1180.51  3467.6 1179.98  3817.4 1155.94  4211.2 1149.24
  4374.6 1149.89  4737.1 1148.91  4813.7 1140.36  4838.2 1134.07  4928.9 1122.37
  4974.8 1123.44  5077.1 1120.94  5079.8 1120.44  5083.1 1120.94  5113.3 1132.53
  5120.4 1135.24  5170.8 1132.31  5211.9 1140.66  5439.8 1148.17  5563.9 1151.15
  5677.2 1159.73  5723.2 1154.22  5840.6 1157.66  5961.5 1157.34  6392.2 1167.76
  6443.5 1168.58  6502.6  1169.1  6566.6 1176.08  6609.9 1196.57  6921.3 1279.88
#Mann= 20 ,-1 , 0
  3361.6      .1       0  3441.6     .05       0  3467.6      .1       0
  3817.4     .16       0  4211.2     .05       0  4374.6      .1       0
  4737.1     .05       0  4813.7      .1       0  4974.8     .05       0
  5077.1     .04       0  5083.1     .05       0  5113.3      .1       0
  5211.9     .16       0  5439.8     .05       0  5563.9     .08       0
  5840.6     .05       0  5961.5      .1       0  6392.2     .16       0
  6443.5     .05       0  6502.6     .16       0
#XS Ineff= 2 ,-1
 5131.31  5220.5 1136.18 5372.07  5549.2 1149.15
Permanent Ineff=
       T       T
Bank Sta=4838.2,5120.4
XS Rating Curve= 0 ,0
Exp/Cntr=0.3,0.1

Type RM Length L Ch R = 1 ,67307   ,851,851,851
BEGIN DESCRIPTION:
MILLER CREEK 100.0
END DESCRIPTION:
XS GIS Cut Line= 4
      2927992.65     10042842.27      2928846.84     10041765.84
       2929277.4     10040356.12      2929638.48     10040196.41
#Sta/Elev= 30
    3031  1180.2  3085.9 1180.17  3128.4 1179.68  3269.5 1176.07  3611.3 1154.49
  3689.2 1147.13  3966.8  1146.1  4679.2  1147.1    4840 1132.75  4856.9 1129.68
  5011.4 1117.26  5014.2 1116.76  5017.4 1117.26    5087 1133.66  5134.3 1138.73
  5210.4  1145.4  5390.4 1159.58  5554.9 1172.52  5590.1 1181.65  5658.6 1179.57
  5734.5    1183  5819.6 1187.63  5891.3 1193.47  5956.9 1204.11  5995.7 1216.65
  6071.1 1231.46  6094.4 1243.53  6146.4  1256.7    6193 1274.22    6274 1286.62
#Mann= 14 ,-1 , 0
    3031      .1       0  3085.9     .16       0  3128.4      .1       0
  3611.3     .16       0  3966.8     .05       0  4856.9      .1       0
  5011.4     .07       0  5017.4      .1       0  5134.3     .05       0
  5210.4     .16       0  5390.4     .05       0  5590.1     .08       0
  5734.5     .05       0  5819.6      .1       0
#XS Ineff= 2 , 0
          4644.6 1147.81
Permanent Ineff=
       T       T
Bank Sta=4840,5087
XS Rating Curve= 0 ,0
Exp/Cntr=0.3,0.1

Type RM Length L Ch R = 1 ,66456   ,596,596,596
BEGIN DESCRIPTION:
MILLER CREEK 99.0
END DESCRIPTION:
XS GIS Cut Line= 3
      2928673.24     10043210.28      2929485.73     10041842.23
      2930138.49     10041203.37
#Sta/Elev= 30
  3143.3 1177.28  3270.7 1174.93  3393.8 1171.69  3415.3 1168.16  3473.7 1150.68
  3582.9 1141.69  3688.3 1139.56  3765.4  1139.7  3828.7 1139.96  4712.8 1144.43
  4820.2 1139.44  4897.9 1129.91  4905.9 1128.95  5008.1 1114.86  5010.8 1114.36
  5014.1 1114.86  5060.5 1120.62    5140 1124.18  5166.7 1125.67  5173.7 1129.21
  5180.8 1132.73    5202 1152.64  5237.4 1155.98  5258.5 1165.69    5293 1167.13
  5331.6 1172.04  5477.9 1182.31  5539.2 1194.17  5569.7  1199.8  5647.8 1204.66
#Mann= 13 ,-1 , 0
  3143.3     .05       0  3270.7     .16       0  3582.9      .1       0
  3688.3     .05       0  3765.4      .1       0  3828.7     .05       0
  4905.9      .1       0  5008.1     .07       0  5014.1      .1       0
    5140     .05       0    5293     .16       0  5331.6      .1       0
  5539.2     .05       0
#XS Ineff= 2 , 0
         4718.18 1144.46
Permanent Ineff=
       T       T
Bank Sta=4897.9,5173.7
XS Rating Curve= 0 ,0
Exp/Cntr=0.3,0.1

Type RM Length L Ch R = 1 ,65860   ,878,878,878
BEGIN DESCRIPTION:
MILLER CREEK 97.0
END DESCRIPTION:
XS GIS Cut Line= 3
      2929041.28     10043425.57      2929846.84     10042307.51
      2930707.98     10041508.88
#Sta/Elev= 30
  3306.7 1174.18  3679.8 1163.32  3807.3 1157.41    3822 1152.91  3842.9 1151.69
  3854.3 1146.07  3887.1 1139.87  3922.7 1138.63  4112.5 1137.92  4724.1 1139.61
  4886.8 1126.31  4939.6 1119.88  4957.6 1115.53  5011.3 1115.14    5014 1114.64
  5017.3 1115.14  5107.3 1121.18  5127.2  1124.6  5162.9 1122.34    5177  1127.1
  5238.7 1143.79  5267.6 1145.17  5377.1 1147.28  5417.4 1152.15  5466.8 1174.99
  5523.5 1196.75  5587.1 1202.39  5637.8 1211.87    5813 1217.73  5859.2 1220.06
#Mann= 13 ,-1 , 0
  3306.7     .16       0  3679.8      .1       0  3854.3     .16       0
  4112.5     .05       0  4939.6     .16       0  5011.3     .07       0
  5017.3     .16       0  5107.3     .05       0  5238.7     .16       0
  5267.6      .1       0  5377.1     .16       0  5637.8      .1       0
    5813     .05       0
#XS Ineff= 2 , 0
         4713.07 1139.95
Permanent Ineff=
       T       T
Bank Sta=4886.8,5177
XS Rating Curve= 0 ,0
Exp/Cntr=0.3,0.1

Type RM Length L Ch R = 1 ,64982   ,1143,1143,1143
BEGIN DESCRIPTION:
MILLER CREEK 96.0
END DESCRIPTION:
XS GIS Cut Line= 3
      2930034.34     10043967.24      2930680.18     10042876.95
      2931152.42      10041640.8
#Sta/Elev= 30
    3385 1169.14  3579.1  1167.1  3718.6 1164.35  3872.6 1153.17    4019 1147.63
  4324.9 1136.61  4666.6 1134.71  4709.2 1129.35  4776.1 1125.95  4800.9 1119.36
  4837.6 1115.02  4984.5 1114.54  4987.3 1114.04  4990.5 1114.54  5019.6 1115.45
    5041 1119.73  5080.1 1129.55  5111.7 1131.48  5126.7 1130.65  5158.8 1135.21
  5215.3 1134.88  5375.3  1136.2  5422.5 1137.57  5474.3 1143.71  5522.8 1168.53
  5565.6 1194.12  5638.7 1208.07  5733.4 1212.82  5828.9 1218.95  5975.5 1225.91
#Mann= 11 ,-1 , 0
    3385     .16       0  3579.1      .1       0    4019     .05       0
  4984.5    .033       0  4990.5     .05       0  5111.7      .1       0
  5215.3     .05       0  5375.3      .1       0  5422.5     .16       0
  5733.4      .1       0  5828.9     .05       0
Bank Sta=4800.9,5041
XS Rating Curve= 0 ,0
Exp/Cntr=0.3,0.1

Type RM Length L Ch R = 1 ,63839   ,620,620,620
BEGIN DESCRIPTION:
MILLER CREEK 93.0
END DESCRIPTION:
XS GIS Cut Line= 3
       2930923.2     10044036.71      2931701.01     10043328.34
      2932166.29     10041863.07
#Sta/Elev= 30
  3543.4 1155.83  3560.1 1155.04  3699.7 1149.47  4271.1 1131.12  4455.6 1129.37
  4733.6 1131.77  4771.1 1128.45  4820.6 1118.54    4975 1104.25  4977.7 1103.75
    4981 1104.25    5020 1105.13  5062.1 1110.73  5104.2 1117.56  5124.9 1121.66
  5156.3 1121.81  5163.9 1125.81  5177.3    1129  5265.7 1132.81  5502.6 1141.91
  5670.5 1170.53  5817.3 1178.88  5838.3 1183.19  5880.3 1186.28  5917.7 1193.99
  6069.2 1203.21  6079.6 1204.48  6111.1 1216.29  6124.6 1217.15  6132.8 1217.18
#Mann= 10 ,-1 , 0
  3543.4     .16       0  3560.1      .1       0  3699.7     .05       0
    4975    .035       0    4981     .05       0  5062.1      .1       0
  5163.9     .05       0  5265.7      .1       0  5917.7     .05       0
  6124.6      .1       0
#XS Ineff= 2 ,-1
  3543.4 4725.57 1132.14 5131.42 5163.17 1121.87
Permanent Ineff=
       T       T
Bank Sta=4820.6,5104.2
XS Rating Curve= 0 ,0
Exp/Cntr=0.3,0.1

Type RM Length L Ch R = 1 ,63219   ,1357,1357,1357
BEGIN DESCRIPTION:
MILLER CREEK 92.0
END DESCRIPTION:
XS GIS Cut Line= 4
      2930819.02     10044196.41      2931971.84     10043807.51
       2932589.9     10042904.73      2933159.39     10042731.11
#Sta/Elev= 30
  3073.1 1160.37  3294.5 1156.21  3494.6 1149.26  3743.5 1145.36  4220.5 1141.42
  4368.3 1137.33  4526.7 1126.22  4792.8 1125.63  4873.4 1116.22  4966.1 1105.67
    5003 1104.88    5020 1104.65  5022.7 1104.15    5026 1104.65  5139.7 1115.24
  5145.5 1116.69  5175.3 1123.72  5226.1 1128.46  5255.5 1128.08  5428.1 1128.99
  5570.5 1137.71  5601.9  1145.1  5664.6 1177.22  5727.3 1219.22  5769.1 1229.03
  5800.5 1249.58  5854.1 1266.93  5881.7 1271.95  5976.7 1274.22  5979.2 1274.22
#Mann= 11 ,-1 , 0
  3073.1     .16       0  3294.5     .05       0  3494.6      .1       0
  3743.5     .05       0    5003      .1       0    5020    .035       0
    5026      .1       0  5139.7     .05       0  5255.5      .1       0
  5428.1     .16       0  5976.7      .1       0
#XS Ineff= 2 , 0
                         5244.89         1129.29
Permanent Ineff=
       T       T
Bank Sta=4873.4,5145.5
XS Rating Curve= 0 ,0
Exp/Cntr=0.3,0.1

Type RM Length L Ch R = 1 ,61862   ,1523,1523,1523
BEGIN DESCRIPTION:
MILLER CREEK 90.0
END DESCRIPTION:
XS GIS Cut Line= 4
      2930622.57     10044418.04      2932289.26     10044322.56
      2933070.51     10044365.96      2933591.33      10043905.9
#Sta/Elev= 30
  2944.9 1164.81  3047.5 1161.16  3341.4 1157.68  3802.1 1145.71  4200.2 1143.93
    4389 1142.58  4553.4 1135.13  4586.6 1129.12  4619.6 1126.13  4853.9 1121.82
    4944 1110.16  4954.5 1108.82  4994.1 1099.13  5064.2 1103.29  5121.3  1098.2
  5124.1  1097.7  5127.3  1098.2  5174.4 1106.23  5224.5 1107.33  5244.5 1111.56
  5396.8 1121.13  5418.4  1126.1  5458.7 1124.06  5473.3 1127.85  5567.3 1150.52
  5737.2 1170.02  5786.5  1182.5  6027.4 1218.06  6041.6 1217.43  6091.7 1227.23
#Mann= 11 ,-1 , 0
  2944.9     .16       0  3047.5     .05       0  4200.2     .16       0
    4389     .05       0  4586.6      .1       0  4619.6     .05       0
  4954.5      .1       0  5121.3     .07       0  5127.3      .1       0
  5458.7     .05       0  5473.3      .1       0
#XS Ineff= 2 , 0
                         5427.27         1126.26
Permanent Ineff=
       T       T
Bank Sta=4944,5244.5
XS Rating Curve= 0 ,0
Exp/Cntr=0.3,0.1

Type RM Length L Ch R = 1 ,60339   ,1286,1286,1286
BEGIN DESCRIPTION:
MILLER CREEK 88.0
END DESCRIPTION:
XS GIS Cut Line= 4
      2931872.61     10046674.98       2932810.1     10045789.57
      2933712.87     10045390.26      2933877.81     10044192.32
#Sta/Elev= 30
    3264 1209.09  3631.2 1198.59  3797.9 1196.66  3861.1 1193.03  4061.3  1187.3
  4235.6 1153.09  4414.8 1122.55  4805.7 1115.99  4904.4 1105.64  4949.5 1096.73
  4994.6 1089.76  4997.3 1089.26  5000.6 1089.76  5096.2  1100.5  5153.7 1093.76
  5196.2 1103.39  5240.6  1107.3  5293.5 1115.55  5375.6 1116.72  5468.8 1118.77
  5706.1 1135.62  5838.5 1136.65  5839.1 1136.64  6002.2 1138.24  6199.7 1143.17
  6298.4 1146.76  6499.6 1156.49  6614.7 1151.91  6661.3 1154.75  6749.9  1170.4
#Mann= 19 ,-1 , 0
    3264     .16       0  3631.2      .1       0  3797.9     .16       0
  3861.1      .1       0  4235.6     .05       0  4949.5      .1       0
  4994.6     .07       0  5000.6      .1       0  5196.2     .05       0
  5375.6     .16       0  5468.8     .05       0  5706.1      .1       0
  5838.5     .05       0  5839.1      .1       0  6002.2     .16       0
  6199.7     .05       0  6298.4      .1       0  6614.7     .05       0
  6661.3      .1       0
#XS Ineff= 2 , 0
                         5547.73         1128.54
Permanent Ineff=
       T       T
Bank Sta=4904.4,5240.6
XS Rating Curve= 0 ,0
Exp/Cntr=0.3,0.1

Type RM Length L Ch R = 1 ,59053   ,1801,1801,1801
BEGIN DESCRIPTION:
MILLER CREEK 86.0
END DESCRIPTION:
XS GIS Cut Line= 4
      2933573.39     10047391.15      2934026.53     10046896.34
      2934182.78     10045948.42      2933984.87     10044130.72
#Sta/Elev= 30
  3911.8  1206.4  3920.4 1205.91  3921.8 1205.83  4050.2 1196.77  4072.5 1195.04
  4282.3 1186.45  4395.4 1177.85  4551.3 1163.88  4737.4 1159.77  4810.4 1127.32
  4872.8 1104.62  4978.3 1088.34  4997.9 1086.75  5000.7 1086.25  5003.9 1086.75
  5056.2 1087.53    5082 1095.46  5183.6 1104.65  5261.1 1110.01  5392.9 1114.19
  5583.4 1114.33  5644.9 1114.14  6263.9 1119.14  6413.3 1133.46  6443.4 1144.04
  6483.7  1135.3  6546.8 1136.76  6552.2  1136.9  6850.4 1145.32  7371.9 1171.54
#Mann= 20 ,-1 , 0
  3911.8     .05       0  3920.4      .1       0  3921.8     .05       0
  4050.2      .1       0  4072.5     .05       0  4282.3      .1       0
  4395.4     .05       0  4551.3      .1       0  4810.4     .16       0
  4978.3      .1       0  4997.9     .07       0  5003.9      .1       0
  5261.1     .05       0  5392.9      .1       0  5583.4     .05       0
  5644.9      .1       0  6263.9     .16       0  6546.8      .1       0
  6552.2     .05       0  6850.4      .1       0
#XS Ineff= 2 ,-1
 5697.73 5890.91 1114.34 6238.64 6336.36 1121.18
Permanent Ineff=
       T       T
Bank Sta=4872.8,5183.6
XS Rating Curve= 0 ,0
Exp/Cntr=0.3,0.1

Type RM Length L Ch R = 1 ,57252   ,1108,1108,1108
BEGIN DESCRIPTION:
MILLER CREEK 84.0
END DESCRIPTION:
XS GIS Cut Line= 3
      2934490.08     10046714.02      2935083.82     10045359.88
      2934100.09      10043907.7
#Sta/Elev= 30
  3178.4 1133.53  4000.3 1127.83  4002.7  1127.8  4110.3 1120.36    4157 1111.47
  4267.2 1110.44  4383.7 1112.16  4538.3 1107.87  4786.8 1101.17  4822.8 1090.19
  4930.6 1092.77  4979.7 1087.48  4993.5 1086.33  4996.2 1085.83  4999.5 1086.33
  5068.4 1087.97  5111.3 1100.54  5134.2 1104.31  5212.2 1104.43    5320 1122.98
  5363.5  1136.2  5391.9 1134.97  5421.8 1125.34  5608.1 1126.51  5630.7 1140.28
  5713.5 1145.94  5877.3 1153.41  5963.2 1157.09  6263.6 1171.17    6411 1186.89
#Mann= 13 ,-1 , 0
  3178.4      .1       0  4000.3     .16       0  4002.7      .1       0
  4267.2     .16       0  4538.3      .1       0  4979.7     .16       0
  4993.5     .07       0  4999.5     .16       0  5363.5     .05       0
  5608.1     .16       0  5713.5      .1       0  5877.3     .16       0
  5963.2      .1       0
#XS Ineff= 4 ,-1
 4148.96 4160.82 1112.91 4166.01 4337.23 1111.87 4483.99 4541.81 1108.34
 5134.78 5193.34 1104.34
Permanent Ineff=
       T       T       T       T
Bank Sta=4786.8,5111.3
XS Rating Curve= 0 ,0
Exp/Cntr=0.3,0.1

Type RM Length L Ch R = 1 ,56144   ,1513,1513,1513
BEGIN DESCRIPTION:
MILLER CREEK 82.0
END DESCRIPTION:
XS GIS Cut Line= 4
       2934745.3     10046552.57      2935490.07     10045568.22
      2936135.91     10045036.97      2937270.25     10044428.17
#Sta/Elev= 30
  3361.4 1130.09  3942.8 1130.45  4077.4 1125.16  4320.1 1105.25  4442.6 1104.89
  4728.9 1106.05  4860.8 1105.65  4903.9 1093.97  4924.7 1089.25  5084.6 1086.52
  5087.3 1086.02  5090.6 1086.52  5116.2 1093.82  5208.8 1097.94  5576.5  1111.9
  5636.6 1122.54  5695.8 1126.34  5768.2 1134.41  5828.3  1149.9  5910.5 1161.49
    5998 1161.57  6017.7 1177.53  6025.6 1183.93  6093.2  1192.4  6210.5 1200.96
  6419.4 1228.78  6459.6 1230.73  6567.2 1235.32    6645 1245.48  6719.4 1256.54
#Mann= 16 ,-1 , 0
  3361.4      .1       0  3942.8     .05       0  4077.4      .1       0
  4320.1     .16       0  4442.6      .1       0  4728.9     .05       0
  5084.6    .035       0  5090.6     .05       0  5208.8      .1       0
  5695.8     .05       0  5910.5      .1       0  6017.7     .08       0
  6210.5      .1       0  6419.4     .16       0  6459.6      .1       0
    6645     .16       0
Bank Sta=4903.9,5116.2
XS Rating Curve= 0 ,0
Exp/Cntr=0.3,0.1

Type RM Length L Ch R = 1 ,54631   ,508,508,508
BEGIN DESCRIPTION:
MILLER CREEK 80.0
END DESCRIPTION:
XS GIS Cut Line= 4
      2934771.31     10046672.38      2935297.37     10046651.55
      2936557.78     10046922.38      2937823.42     10046854.67
#Sta/Elev= 30
  4035.6 1130.04  4117.5 1126.19  4119.9 1126.01  4202.9 1120.21  4402.9 1123.37
  4463.1 1123.07  4751.5 1100.25  4851.5 1094.68  4878.5 1090.83  4950.2  1078.8
  4969.1 1072.16  4971.9 1071.66  4975.1 1072.16  5026.6 1073.04  5048.5 1078.12
  5196.1 1087.99  5238.3 1090.93  5253.5 1091.58  5312.6 1095.57  5349.6 1107.97
  5391.7 1122.63  5574.4 1129.76  5851.2 1135.43  6003.9 1142.06  6306.9    1153
  6548.6  1164.2  6728.9 1172.01  7063.7 1179.15  7083.7 1186.28  7118.7 1188.21
#Mann= 19 ,-1 , 0
  4035.6      .1       0  4117.5     .05       0  4119.9      .1       0
  4402.9     .05       0  4751.5      .1       0  4851.5     .05       0
  4950.2      .1       0  4969.1     .07       0  4975.1      .1       0
  5048.5     .05       0  5196.1      .1       0  5253.5     .16       0
  5349.6      .1       0  5574.4     .16       0  5851.2      .1       0
  6003.9     .16       0  6306.9      .1       0  6548.6     .16       0
  6728.9      .1       0
Bank Sta=4878.5,5238.3
XS Rating Curve= 0 ,0
Exp/Cntr=0.3,0.1

Type RM Length L Ch R = 1 ,54123   ,1612,1612,1612
BEGIN DESCRIPTION:
MILLER CREEK 79.0
END DESCRIPTION:
XS GIS Cut Line= 4
      2934677.54     10046682.78      2935396.32      10047182.8
      2936125.49      10047370.3      2937807.74     10047000.52
#Sta/Elev= 30
    3926 1130.17  3995.8 1129.19  4170.8    1121  4322.4 1110.27  4653.2 1102.08
  4724.7 1097.55  4822.4 1096.92  4845.1 1094.96  4876.3    1088    4969  1073.8
  5017.6 1073.08  5020.4 1072.58  5023.6 1073.08  5148.8 1084.55  5172.7 1086.98
  5175.5 1087.21  5270.4 1093.33  5299.4  1102.4  5330.4 1119.85  5346.7 1123.09
  5386.8 1124.01  5703.8  1126.7  6038.8 1133.97  6357.4 1148.49    6727 1160.79
  6964.3 1172.63  7103.8 1178.58  7246.9  1178.2  7257.2 1178.76  7276.9 1186.38
#Mann= 11 ,-1 , 0
    3926      .1       0  3995.8     .05       0  4170.8      .1       0
  4876.3     .16       0  5017.6     .07       0  5023.6     .16       0
  5148.8      .1       0  5172.7     .16       0  5386.8      .1       0
    6727     .16       0  6964.3      .1       0
Bank Sta=4876.3,5175.5
XS Rating Curve= 0 ,0
Exp/Cntr=0.3,0.1

Type RM Length L Ch R = 1 ,52511   ,2054,2054,2054
BEGIN DESCRIPTION:
MILLER CREEK 76.0
END DESCRIPTION:
XS GIS Cut Line= 4
      2933823.41     10048318.21      2935099.45     10048286.97
      2935917.16     10047573.42      2937807.78     10047401.55
#Sta/Elev= 30
  4285.2  1206.4  4296.5 1206.25  4395.3 1209.54  4567.3 1222.12  4630.4 1214.76
  4671.7 1193.97  4790.4 1103.43  4840.4 1081.21  4960.5  1063.1  4997.5 1062.59
  5000.2 1062.09  5003.5 1062.59  5040.5  1063.4  5110.5  1081.3  5143.1 1084.16
  5223.6 1092.38    5599 1095.75  5789.8 1114.36  6053.4 1120.58  6087.4 1120.77
  6259.7 1121.64  6286.7 1121.68  6527.4 1120.07  7437.5 1135.92  7651.1 1142.96
  7762.2 1146.92  7840.6 1149.76  8236.9 1164.63  8324.6 1171.92  8545.3 1175.69
#Mann= 20 ,-1 , 0
  4285.2     .05       0  4296.5     .16       0  4395.3     .05       0
  4567.3      .1       0  4671.7     .05       0  4840.4      .1       0
  4997.5     .07       0  5003.5      .1       0  5143.1     .16       0
  5223.6      .1       0  6053.4     .05       0  6087.4      .1       0
  6259.7     .05       0  6286.7      .1       0  7437.5     .16       0
  7651.1      .1       0  7762.2     .16       0  7840.6      .1       0
  8236.9     .16       0  8324.6      .1       0
#XS Ineff= 2 , 0
                         5323.86         1096.05
Permanent Ineff=
       T       T
Bank Sta=4840.4,5110.5
XS Rating Curve= 0 ,0
Exp/Cntr=0.3,0.1

Type RM Length L Ch R = 1 ,50457   ,587,587,587
BEGIN DESCRIPTION:
MILLER CREEK 74.0
END DESCRIPTION:
XS GIS Cut Line= 4
       2934615.1     10049318.22      2935891.12     10049328.63
      2936990.07     10048089.05      2937760.87     10047906.76
#Sta/Elev= 30
  3200.8 1164.94  3384.2 1158.12  3513.9 1145.08  3614.2 1135.46  3994.2 1114.73
    4252 1109.62  4350.7 1104.35  4747.9 1084.01  4828.4 1075.98  4832.3 1075.57
  4917.6 1071.29  5018.6 1058.94  5020.9 1058.18  5023.6 1057.68  5026.9 1058.18
  5052.3 1067.25  5109.2 1075.27  5158.5 1080.36  5208.5 1078.58  5214.4 1078.71
  5271.9 1073.11  5335.2  1091.8  5392.2 1121.29  5456.6 1124.63  5725.6 1137.47
  6228.2 1146.62  6441.9 1153.69  6486.7  1155.1  6721.5 1163.69  6925.5 1173.25
#Mann= 16 ,-1 , 0
  3200.8     .05       0  3513.9      .1       0    4252     .05       0
  4350.7      .1       0  4828.4     .16       0  5018.6      .1       0
  5020.9     .07       0  5026.9      .1       0  5208.5     .05       0
  5214.4      .1       0  5335.2     .16       0  5456.6      .1       0
  6228.2     .16       0  6441.9      .1       0  6486.7     .16       0
  6721.5      .1       0
#XS Ineff= 2 , 0
                         5172.73         1080.65
Permanent Ineff=
       T       T
Bank Sta=4832.3,5109.2
XS Rating Curve= 0 ,0
Exp/Cntr=0.3,0.1

Type RM Length L Ch R = 1 ,49870   ,1272,1272,1272
BEGIN DESCRIPTION:
MILLER CREEK 73.0
END DESCRIPTION:
XS GIS Cut Line= 4
      2934708.86     10049448.43      2935917.16     10049609.88
      2937271.32     10049146.34       2938359.9       10049063.
#Sta/Elev= 30
  3037.7 1153.11  3531.7 1123.66  3895.1 1114.82    3993 1114.92    4092 1113.07
  4180.8 1111.74  4262.4 1109.57    4398 1099.87  4503.9 1086.37  4609.7 1085.27
  4882.4 1073.38  4927.2 1067.15  5025.3 1058.13  5028.1 1057.63  5031.3 1058.13
  5138.8 1073.97  5153.5 1092.87  5209.4 1121.57  5244.6 1123.94  5350.5  1127.3
  5409.5 1129.71  5829.5 1150.72  5986.1 1158.56  6136.5 1180.66  6229.7 1168.66
  6407.3 1168.56  6427.3 1182.66  6463.4 1185.01  6562.7 1190.78  6779.8 1204.91
#Mann= 20 ,-1 , 0
  3037.7      .1       0  3895.1     .16       0    3993      .1       0
    4092     .05       0  4180.8      .1       0  4262.4     .05       0
    4398      .1       0  4503.9     .16       0  4609.7      .1       0
  4927.2     .05       0  5025.3    .035       0  5031.3     .05       0
  5138.8     .16       0  5244.6      .1       0  5350.5     .05       0
  5409.5      .1       0  5829.5     .05       0  6229.7      .1       0
  6463.4     .05       0  6562.7      .1       0
Bank Sta=4882.4,5138.8
XS Rating Curve= 0 ,0
Exp/Cntr=0.3,0.1

Type RM Length L Ch R = 1 ,48598   ,1037,1037,1037
BEGIN DESCRIPTION:
MILLER CREEK 71.0
END DESCRIPTION:
XS GIS Cut Line= 3
      2934745.27     10049854.67      2937010.91     10050875.51
      2937993.89     10051598.44
#Sta/Elev= 30
  3631.2 1134.55  4144.3 1116.02  4385.8 1111.66  4448.1 1108.84  4471.3 1101.96
    4492 1107.61  4525.2  1109.2  4843.2  1101.7  4874.1  1092.4    4918 1069.66
  4939.9 1059.21  5004.7 1058.03  5007.5 1057.53  5010.7 1058.03  5324.4 1070.32
  5342.7 1071.46  5394.4 1077.94  5440.7 1094.22  5538.8 1116.75    5660 1119.65
  5798.6 1122.93    6033 1127.06  6390.2 1134.49  6641.4 1146.57  6674.7 1148.14
  6817.6 1150.09  6958.8 1152.67  6979.2 1161.66  7064.8 1172.31  7336.4  1181.9
#Mann= 17 ,-1 , 0
  3631.2      .1       0  4144.3     .16       0  4385.8      .1       0
    4492     .16       0  4525.2     .05       0  4843.2      .1       0
  5004.7     .07       0  5010.7      .1       0  5324.4     .16       0
    5660     .05       0  5798.6      .1       0    6033     .05       0
  6390.2      .1       0  6641.4     .05       0  6674.7      .1       0
  6817.6     .05       0  6958.8      .1       0
#XS Ineff= 2 , 0
         4788.64 1106.28
Permanent Ineff=
       T       T
Bank Sta=4918,5342.7
XS Rating Curve= 0 ,0
Exp/Cntr=0.3,0.1

Type RM Length L Ch R = 1 ,47561   ,916,916,916
BEGIN DESCRIPTION:
MILLER CREEK 70.0
END DESCRIPTION:
XS GIS Cut Line= 2
      2934612.44     10050003.51      2936604.47     10052162.12
#Sta/Elev= 30
  3135.2 1134.83  3592.6  1124.7  3745.6 1115.68  4052.5 1100.26  4179.8 1101.85
  4223.3 1103.05  4301.8  1100.5  4503.9 1092.41    4525 1094.46  4692.9 1080.34
  4827.3 1066.04  4845.2 1064.77  4951.2 1058.22  4972.5 1049.61  5004.6 1048.02
  5011.7 1047.45  5014.5 1046.95  5017.7 1047.45  5043.1 1059.23  5085.6 1064.81
  5099.8 1071.51  5135.5  1101.8  5170.7  1111.6  5203.8 1113.33  5490.4 1128.35
  5602.2 1133.97  5810.6 1156.66  5829.8 1157.29  5941.9 1161.94  6072.5 1178.07
#Mann= 16 ,-1 , 0
  3135.2      .1       0  3745.6     .16       0  4179.8      .1       0
  4223.3     .05       0  4301.8      .1       0  4503.9     .16       0
    4525      .1       0  4692.9     .16       0  4827.3      .1       0
  5004.6     .16       0  5011.7     .07       0  5017.7     .16       0
  5203.8      .1       0  5490.4     .05       0  5810.6      .1       0
  5829.8     .05       0
Bank Sta=4845.2,5085.6
XS Rating Curve= 0 ,0
Exp/Cntr=0.3,0.1

Type RM Length L Ch R = 1 ,46645   ,603,603,603
BEGIN DESCRIPTION:
MILLER CREEK 69.0
END DESCRIPTION:
XS GIS Cut Line= 3
      2934418.02     10050239.64      2935216.64     10052031.32
      2936022.15     10052274.37
#Sta/Elev= 30
  3292.9 1135.22  3848.5 1123.54  4055.8 1105.59  4206.9 1101.37  4234.8 1101.28
  4316.7 1098.03  4426.5  1093.7    4456 1093.42  4536.2 1092.56  4695.9 1079.92
    4863 1063.95  4916.3 1060.09    5003 1045.16  5005.7 1044.66    5009 1045.16
  5119.6 1053.58  5150.8 1056.27  5158.6 1062.17  5180.5 1076.27  5202.7 1082.73
  5243.7 1084.83  5352.5 1102.23  5535.9 1111.71  5684.7 1117.49    5716 1125.13
  5818.6 1132.79  5862.3  1134.8  5935.9 1150.94  6017.5 1162.25  6095.9 1172.62
#Mann= 17 ,-1 , 0
  3292.9      .1       0  4055.8     .16       0  4206.9      .1       0
  4234.8     .16       0  4316.7      .1       0  4426.5     .05       0
    4456      .1       0  4536.2     .05       0  4695.9     .16       0
  4916.3     .05       0    5003    .035       0    5009     .05       0
  5119.6      .1       0  5535.9     .05       0  5818.6      .1       0
  5935.9     .05       0  6017.5      .1       0
Bank Sta=4863,5158.6
XS Rating Curve= 0 ,0
Exp/Cntr=0.3,0.1

Type RM Length L Ch R = 1 ,46042   ,541,541,541
BEGIN DESCRIPTION:
MILLER CREEK 68.0
END DESCRIPTION:
XS GIS Cut Line= 4
      2933841.63     10050135.48      2934230.53     10051392.43
      2934681.91     10052274.38       2936022.2     10052364.66
#Sta/Elev= 30
  2974.6 1147.71  4200.8 1122.13    4608 1107.32  4702.2 1090.42  4780.1 1077.54
  4824.5 1061.99  4893.7 1044.96  4957.7 1049.68  5007.7 1043.38  5010.5 1042.88
  5013.7 1043.38  5040.9 1054.06  5092.9 1054.45  5253.3 1059.23  5287.6 1062.99
  5350.6  1070.3  5449.2 1075.29    5509  1078.6  5676.4  1085.2  5714.1 1090.52
  5914.8 1106.92  5997.2 1110.79  6099.5 1114.54  6169.6 1128.34  6262.6  1132.4
    6308 1135.41  6400.2 1156.38  6510.4 1168.92  6560.5 1181.19  6624.4 1183.44
#Mann= 16 ,-1 , 0
  2974.6      .1       0  4702.2     .16       0  4893.7      .1       0
  5007.7     .07       0  5013.7      .1       0  5092.9     .05       0
  5253.3     .16       0  5350.6      .1       0  5449.2     .05       0
    5509      .1       0  5676.4     .16       0  5714.1      .1       0
  5914.8     .05       0  5997.2      .1       0  6262.6     .05       0
    6308      .1       0
Bank Sta=4824.5,5287.6
XS Rating Curve= 0 ,0
Exp/Cntr=0.3,0.1

Type RM Length L Ch R = 1 ,45501   ,320,320,320
BEGIN DESCRIPTION:
MILLER CREEK 67.0
END DESCRIPTION:
XS GIS Cut Line= 3
      2932723.54      10051718.8      2933869.41     10052406.32
      2936063.63      10052434.1
#Sta/Elev= 30
  3301.1 1179.03    3434 1171.93  3592.5 1168.98  3746.1 1151.28  3896.4 1146.02
  4102.8 1141.87  4584.9 1130.64  4696.5 1115.73  4856.5 1090.07  4926.5  1071.2
 4940.91 1061.63  4966.5 1045.14  4993.5 1044.13  4996.2 1043.63  4999.5 1044.13
  5026.5 1051.93  5196.5 1053.67  5316.2 1061.47  5346.5 1062.92  5414.8 1068.06
  5513.4  1073.6    5612 1077.99  5809.3 1084.52    5891 1093.67  6047.4 1105.88
  6238.2 1115.74  6306.6 1128.19  6436.6 1136.02  6676.6 1181.05  6831.8 1191.15
#Mann= 16 ,-1 , 0
  3301.1     .05       0    3434      .1       0  3896.4     .05       0
  4102.8      .1       0  4584.9     .05       0  4696.5      .1       0
  4993.5     .07       0  4999.5      .1       0  5316.2     .16       0
  5414.8      .1       0  5513.4     .16       0    5612     .05       0
  5809.3     .16       0    5891      .1       0  6047.4     .05       0
  6238.2      .1       0
Bank Sta=4940.91,5346.5
XS Rating Curve= 0 ,0
Exp/Cntr=0.3,0.1

Type RM Length L Ch R = 1 ,45181   ,566,566,566
BEGIN DESCRIPTION:
MILLER CREEK 66.0
END DESCRIPTION:
XS GIS Cut Line= 4
      2933098.55     10052711.88      2934036.08     10052767.43
      2934987.47     10052607.71      2935924.21     10052545.26
#Sta/Elev= 30
  3821.8  1160.3  3919.2 1151.79  4394.2 1136.36    4563 1130.63  4623.1 1119.16
  4725.8 1112.87  4844.5 1098.98  4895.2 1076.96  4915.5 1061.84  4932.5 1047.05
  4990.1 1042.62  4992.9 1042.12  4996.1 1042.62  5037.2 1050.24    5169 1061.53
  5243.4 1066.18  5373.3 1071.41  5471.1 1073.21  5489.9 1074.28  5570.9  1078.4
  5771.7 1084.85  5870.8 1096.18  5997.9 1104.52  6137.6 1110.53  6218.6 1126.21
  6388.1  1137.3  6468.3  1156.1  6558.5 1167.16    6608 1179.31  6664.5 1182.39
#Mann= 15 ,-1 , 0
  3821.8     .16       0  3919.2      .1       0  4394.2     .05       0
  4725.8      .1       0  4990.1     .07       0  4996.1      .1       0
  5243.4     .05       0  5373.3      .1       0  5471.1     .05       0
  5489.9     .16       0  5570.9     .05       0  5771.7      .1       0
  5870.8     .16       0  5997.9     .05       0  6218.6      .1       0
Bank Sta=4915.5,5169
XS Rating Curve= 0 ,0
Exp/Cntr=0.3,0.1

Type RM Length L Ch R = 1 ,44615   ,516,516,516
BEGIN DESCRIPTION:
MILLER CREEK 65.0
END DESCRIPTION:
XS GIS Cut Line= 4
      2933168.03     10053204.93      2934348.58     10053316.04
      2934987.47     10052927.16      2935862.51      10052670.2
#Sta/Elev= 30
  3610.5 1146.33  3773.1 1143.02  3970.5 1137.52  4071.3  1133.7  4123.2 1131.43
  4201.3 1117.47  4340.2 1105.96  4414.5 1102.85  4476.7 1090.89  4591.8 1076.34
  4719.5  1071.3  4776.1 1059.03  4788.5  1057.7  4808.7 1055.15  4925.3 1048.31
  5014.3 1040.47  5017.1 1039.97  5020.3 1040.47  5088.8 1059.73  5118.1 1068.14
  5189.6 1067.98  5215.7 1066.15  5340.8 1070.87  5663.7 1092.85  5786.4 1099.88
  5965.9 1106.98  6048.3 1121.19  6233.1 1133.87    6354 1157.65  6456.2  1165.8
#Mann= 19 ,-1 , 0
  3610.5      .1       0  3773.1     .16       0  3970.5      .1       0
  4071.3     .05       0  4201.3      .1       0  4340.2     .05       0
  4476.7      .1       0  4591.8     .05       0  4788.5      .1       0
  4808.7     .05       0  4925.3      .1       0  5014.3     .07       0
  5020.3      .1       0  5189.6     .05       0  5215.7      .1       0
  5340.8     .05       0  5663.7      .1       0  5786.4     .05       0
  6048.3      .1       0
Bank Sta=4776.1,5088.8
XS Rating Curve= 0 ,0
Exp/Cntr=0.3,0.1

Type RM Length L Ch R = 1 ,44099   ,855,855,855
BEGIN DESCRIPTION:
MILLER CREEK 64.0
END DESCRIPTION:
XS GIS Cut Line= 3
      2933751.38      10054468.8      2935265.25     10053267.43
      2935931.56     10052788.52
#Sta/Elev= 30
  3646.7 1147.84    3741 1135.47  4003.8 1126.48    4091 1111.98  4146.4 1110.06
  4268.2 1091.26  4391.3 1083.66  4453.5 1079.48  4691.7 1069.46  4714.2 1064.05
    4752 1058.02  4841.9 1052.82  4845.9 1052.64  4929.9 1047.17  4941.3 1043.36
    4991 1040.52  4993.7 1040.02    4997 1040.52  5122.1 1058.57  5144.2 1060.63
  5292.5 1076.58  5442.7 1080.81  5593.7 1086.39  5885.3 1110.88  5950.3  1121.7
  5999.5  1124.6  6087.5 1128.26  6172.5 1131.69  6264.6 1147.41  6399.9 1159.29
#Mann= 17 ,-1 , 0
  3646.7     .05       0    4091     .16       0  4391.3     .05       0
  4453.5     .16       0  4691.7      .1       0  4714.2     .05       0
  4841.9      .1       0  4845.9     .05       0  4941.3      .1       0
    4991     .07       0    4997      .1       0  5144.2     .05       0
  5292.5      .1       0  5442.7     .05       0  5593.7      .1       0
  5999.5     .05       0  6087.5      .1       0
Bank Sta=4752,5122.1
XS Rating Curve= 0 ,0
Exp/Cntr=0.3,0.1

Type RM Length L Ch R = 1 ,43244   ,795,795,795
BEGIN DESCRIPTION:
MILLER CREEK 63.0
END DESCRIPTION:
XS GIS Cut Line= 4
      2934640.22     10054975.79      2935223.58      10054559.1
      2935598.58     10053857.71      2936015.25     10052934.09
#Sta/Elev= 30
  3884.4 1123.45  3978.5 1119.91  4129.6 1101.26  4160.5 1099.16  4278.3 1091.96
  4379.7 1080.73  4623.3  1065.4  4687.8 1066.22  4743.5 1066.41 4795.45 1055.22
  4822.8    1047  4875.3 1048.19  4913.5 1045.31  4924.9 1038.37  4963.2 1038.57
  4998.3 1036.34  5001.1 1035.84  5004.3 1036.34  5029.7 1043.93    5133 1055.56
  5141.5  1056.1    5259 1062.43    5363 1076.47  5719.1 1095.02  5869.9 1109.57
  5915.2 1115.42  6043.7 1119.67  6260.9 1132.52  6388.9  1146.5  6409.9 1148.23
#Mann= 13 ,-1 , 0
  3884.4     .16       0  4129.6      .1       0  4160.5     .16       0
  4379.7      .1       0  4687.8     .16       0  4963.2      .1       0
  4998.3     .07       0  5004.3      .1       0  5029.7     .16       0
  5141.5      .1       0  5869.9     .05       0  6043.7      .1       0
  6388.9     .16       0
#XS Ineff= 2 , 0
         4727.27 1068.01
Permanent Ineff=
       T       T
Bank Sta=4795.45,5133
XS Rating Curve= 0 ,0
Exp/Cntr=0.3,0.1

Type RM Length L Ch R = 1 ,42449   ,632,632,632
BEGIN DESCRIPTION:
MILLER CREEK 62.0
END DESCRIPTION:
XS GIS Cut Line= 3
      2934668.06     10055052.15      2935869.41     10054899.38
      2936966.62     10053441.07
#Sta/Elev= 30
  3462.8 1122.89  3513.6 1121.64    3751 1098.34  3927.4 1085.74  4603.5 1062.48
  4705.9 1053.92    4767  1048.6  4819.2 1039.99  4843.4 1044.79  4933.7 1043.29
  4962.6 1037.13  5003.3 1034.44    5006 1033.94  5009.3 1034.44  5056.3 1046.68
  5119.1 1054.06  5201.2  1058.5  5248.2 1061.03  5288.9 1069.04  5383.5 1097.04
  5439.8 1103.58  5462.7 1109.19  5569.4 1117.42  5706.3 1122.65  5792.8 1125.69
  5816.2 1127.24  6038.9 1138.31  6297.7 1157.62  6383.1    1172  6498.8  1177.6
#Mann= 15 ,-1 , 0
  3462.8     .16       0    3751      .1       0  3927.4     .05       0
    4767      .1       0  4843.4     .05       0  4962.6     .16       0
  5003.3     .07       0  5009.3     .16       0  5201.2      .1       0
  5288.9     .16       0  5439.8      .1       0  5706.3     .16       0
  5792.8      .1       0  5816.2     .05       0  6038.9      .1       0
Bank Sta=4705.9,5119.1
XS Rating Curve= 0 ,0
Exp/Cntr=0.3,0.1

Type RM Length L Ch R = 1 ,41817   ,759,759,759
BEGIN DESCRIPTION:
MILLER CREEK 61.0
END DESCRIPTION:
XS GIS Cut Line= 3
      2935098.63     10055225.76      2936049.97     10055177.16
      2937258.28     10054850.77
#Sta/Elev= 30
  3571.1 1089.43  3591.6 1088.06  3647.3  1085.9  3891.4 1083.13  4041.6 1070.27
  4071.6 1071.07  4291.8 1060.74  4512.2 1058.07  4603.5 1053.31  4631.8 1051.89
  4739.7  1045.6    4791 1040.56  4812.2 1040.09  4843.2 1043.81  4894.4 1045.08
  4898.2 1044.91  4926.1 1044.39  4975.3 1036.33  4995.6 1035.21  4998.4 1034.71
  5001.6 1035.21  5020.3 1037.33    5040 1044.25 5046.88 1051.54    5055 1058.64
  5081.5 1088.35  5131.1    1113    5154 1115.11  5728.4  1126.1  5775.3 1127.77
#Mann= 11 ,-1 , 0
  3571.1     .16       0  3591.6      .1       0  3647.3     .05       0
  4603.5      .1       0    4791     .05       0  4894.4      .1       0
  4898.2     .16       0  4995.6     .07       0  5001.6     .16       0
  5131.1      .1       0  5728.4     .05       0
Bank Sta=4631.8,5046.88
XS Rating Curve= 0 ,0
Exp/Cntr=0.3,0.1

Type RM Length L Ch R = 1 ,41058   ,581,581,581
BEGIN DESCRIPTION:
MILLER CREEK 60.0
END DESCRIPTION:
XS GIS Cut Line= 4
      2935070.84     10055309.11       2936070.8     10055510.49
       2936633.3     10055989.66       2937097.3     10056058.91
#Sta/Elev= 30
  3624.4 1090.79  3669.6 1087.68  3769.3 1085.05  4070.8  1080.8  4213.6 1071.59
  4387.2 1071.68  4509.4 1061.36  4621.7 1056.93  4798.4 1055.39  4822.7 1055.56
  4843.6 1049.26  4876.3 1044.01  4900.7 1044.72  4923.4 1037.25  4929.3 1034.41
  5004.2 1033.99    5007 1033.49  5010.2 1033.99  5011.5 1034.17  5120.3 1038.93
    5206 1050.71  5290.5 1072.68  5304.8  1082.2  5339.9 1087.55  5382.6 1099.62
  5398.7 1109.23  5418.9 1115.64  5600.9 1132.53  5712.7 1136.04  5852.5 1144.96
#Mann= 10 ,-1 , 0
  3624.4     .16       0  3669.6      .1       0  3769.3     .05       0
  4798.4      .1       0  4876.3     .16       0  4923.4      .1       0
  5004.2     .07       0  5010.2      .1       0  5011.5     .16       0
  5712.7      .1       0
#XS Ineff= 2 , 0
         4708.81 1057.85
Permanent Ineff=
       T       T
Bank Sta=4843.6,5206
XS Rating Curve= 0 ,0
Exp/Cntr=0.3,0.1

Type RM Length L Ch R = 1 ,40477   ,894,894,894
BEGIN DESCRIPTION:
MILLER CREEK 59.0
END DESCRIPTION:
XS GIS Cut Line= 3
       2934980.5      10055593.8      2935966.64     10056239.66
      2936918.02     10056239.66
#Sta/Elev= 30
  3609.9    1098  3752.8 1088.08  3884.1 1079.78  4041.5 1073.86  4336.6 1067.54
  4626.1 1064.45  4698.5  1061.7  4785.5 1053.73  4870.5 1054.96  4930.5 1048.03
  4950.5 1043.27  4960.5 1037.67  4977.5 1034.68  4980.3 1034.18  4983.5 1034.68
  4999.8 1034.98  5050.5 1034.75  5070.5 1038.66  5110.5 1036.26  5200.5 1037.68
  5232.1 1041.72  5320.5 1047.53  5360.5 1053.89  5410.5 1083.13  5430.5 1091.37
  5480.5 1118.21  5570.5 1126.02  5600.5 1133.42  5660.5 1135.62  5740.1 1142.96
#Mann= 10 ,-1 , 0
  3609.9     .16       0  3752.8     .05       0  3884.1      .1       0
  4041.5     .05       0  4336.6      .1       0  4785.5     .05       0
  4977.5     .07       0  4983.5     .05       0  4999.8      .1       0
  5232.1     .16       0
#XS Ineff= 2 , 0
         4859.38 1055.22
Permanent Ineff=
       T       T
Bank Sta=4930.5,5320.5
XS Rating Curve= 0 ,0
Exp/Cntr=0.3,0.1

Type RM Length L Ch R = 1 ,39583   ,1004,1004,1004
BEGIN DESCRIPTION:
MILLER CREEK 58.0
END DESCRIPTION:
XS GIS Cut Line= 4
      2935327.76     10057878.54      2936091.64     10057163.27
      2936654.14     10057045.21      2936959.41      10056788.5
#Sta/Elev= 30
  3656.7 1099.39  3802.1 1094.31  3887.1 1087.45  3956.2 1077.87  4049.8  1067.1
  4102.2 1065.29    4143 1064.62  4205.6 1061.59  4323.9 1061.21  4464.7 1060.27
    4561 1059.17  4636.9 1050.89  4825.1 1050.82  4863.4 1043.99  4869.9 1037.03
  4885.9 1034.22  4961.6 1028.38  4964.3 1027.88  4967.6 1028.38  5006.5 1028.68
  5039.5 1035.57  5141.2 1040.45  5180.2 1044.54  5200.6  1047.3  5237.9 1063.66
  5309.9 1085.94  5395.7 1104.17  5445.1 1117.76    5609 1127.75  5676.8  1136.3
#Mann= 13 ,-1 , 0
  3656.7     .16       0  3956.2     .05       0  4102.2      .1       0
    4143     .05       0  4323.9      .1       0  4464.7     .16       0
    4561     .05       0  4885.9      .1       0  4961.6     .07       0
  4967.6      .1       0  5039.5     .16       0  5141.2     .05       0
  5237.9     .16       0
Bank Sta=4863.4,5180.2
XS Rating Curve= 0 ,0
Exp/Cntr=0.3,0.1

Type RM Length L Ch R = 1 ,38579   ,504,504,504
BEGIN DESCRIPTION:
MILLER CREEK 57.0
END DESCRIPTION:
XS GIS Cut Line= 4
      2936140.26     10058850.75      2936612.47     10058156.32
       2936883.3      10057871.6      2937098.57     10056871.63
#Sta/Elev= 30
  3979.2 1095.76    4127 1090.09  4265.7 1077.15  4369.4 1071.74  4552.6 1063.58
  4710.6 1057.61  4746.5 1047.17  4788.5 1041.78  4846.3 1034.49    4903 1031.69
    4921 1027.99  4923.8 1027.49    4927 1027.99  4977.4 1028.36  5023.1  1028.8
  5058.5 1032.67  5107.9 1039.52  5129.1 1041.93    5220 1048.52    5457 1055.97
  5532.6 1057.33  5721.2 1062.36  5751.9 1061.07  5878.8 1072.82    5930 1084.96
  6021.7 1101.66  6065.9 1116.18  6115.3 1120.75  6164.6 1121.56  6234.8 1130.84
#Mann= 12 ,-1 , 0
  3979.2     .16       0  4265.7      .1       0  4369.4     .05       0
  4552.6      .1       0    4921    .033       0    4927      .1       0
  4977.4     .05       0  5058.5     .16       0  5107.9      .1       0
    5457     .05       0  5532.6      .1       0    5930     .16       0
Bank Sta=4788.5,5129.1
XS Rating Curve= 0 ,0
Exp/Cntr=0.3,0.1
