--- SYCAMORE CREEK.prj (project) ---

Proj Title=SYCAMORE CREEK Base Level Engineering
Current Plan=p01
Default Exp/Contr=0.3,0.1
English Units
Geom File=g01
Flow File=f01
Plan File=p01
Y Axis Title=Elevation
X Axis Title(PF)=Main Channel Distance
X Axis Title(XS)=Station
BEGIN DESCRIPTION:
SYCAMORE CREEK
END DESCRIPTION:
DSS Export Rating Curves= 0
DSS Export Rating Curve Sorted= 0
DSS Export Volume Flow Curves= 0
DXF OffsetX= 0
DXF OffsetY= 0
DXF ScaleX= 1
DXF ScaleY= 10

--- SYCAMORE CREEK.p01 (plan) ---

Plan Title=Multiple Run
Short Identifier=Multiple
Geom File=g01
Flow File=f01
Subcritical Flow
K Sum by GR= 0
Std Step Tol= 0.01
Critical Tol= 0.01
Num of Std Step Trials= 20
Max Error Tol= 0.3
Flow Tol Ratio= 0.001
Split Flow NTrial= 30
Split Flow Tol= 0.02
Split Flow Ratio= 0.02
Log Output Level= 0
Friction Slope Method= 1
Unsteady Friction Slope Method= 2
Unsteady Bridges Friction Slope Method= 1
Parabolic Critical Depth
Global Vel Dist=  1 , 1 , 1
Global Log Level= 0
CheckData=True
Encroach Param= -1, 0, 0, 0
BEGIN DESCRIPTION:
Multiple Run
END DESCRIPTION:

--- SYCAMORE CREEK.f01 (steady flow) ---

Flow Title=Multiple
Program Version=4.10
Number of Profiles= 7
Profile Names=10-year,25-year,50-year,1pct_min,100-year,1pct_plu,500-year
River Rch & RM=SYCAMORE CREEK,Reach-1         ,22276
     975    1423    1816    1697    2296    3104    3679
River Rch & RM=SYCAMORE CREEK,Reach-1         ,19593
    1588    2382    3096    2942    3979    5382    6599
River Rch & RM=SYCAMORE CREEK,Reach-1         ,18006
    2105    3197    4189    4011    5424    7335    9129
River Rch & RM=SYCAMORE CREEK,Reach-1         ,14524
    2395    3650    4793    4596    6215    8405   10492
River Rch & RM=SYCAMORE CREEK,Reach-1         ,9408
    3237    4999    6623    6401    8656   11707   14850
River Rch & RM=SYCAMORE CREEK,Reach-1         ,6797
    4794    7502   10027    9764   13205   17859   23002
Boundary for River Rch & Prof#=SYCAMORE CREEK,Reach-1         , 1
Up Type= 0
Dn Type= 3
Dn Slope=0.013
Boundary for River Rch & Prof#=SYCAMORE CREEK,Reach-1         , 2
Up Type= 0
Dn Type= 3
Dn Slope=0.013
Boundary for River Rch & Prof#=SYCAMORE CREEK,Reach-1         , 3
Up Type= 0
Dn Type= 3
Dn Slope=0.013
Boundary for River Rch & Prof#=SYCAMORE CREEK,Reach-1         , 4
Up Type= 0
Dn Type= 3
Dn Slope=0.013
Boundary for River Rch & Prof#=SYCAMORE CREEK,Reach-1         , 5
Up Type= 0
Dn Type= 3
Dn Slope=0.013
Boundary for River Rch & Prof#=SYCAMORE CREEK,Reach-1         , 6
Up Type= 0
Dn Type= 3
Dn Slope=0.013
Boundary for River Rch & Prof#=SYCAMORE CREEK,Reach-1         , 7
Up Type= 0
Dn Type= 3
Dn Slope=0.013
DSS Import GetInterval= 0
DSS Import GetPeak= 0
DSS Import FillOption= 0

--- SYCAMORE CREEK.g01 (geometry) ---

Geom Title=Existing Conditions
Program Version=4.10

River Reach=SYCAMORE CREEK  ,Reach-1
Reach XY= 30
      2968920.29     10053704.29      2968547.09     10054411.16
      2967924.04     10054431.16      2968056.72     10054907.75
      2967499.06     10056038.34      2967777.41     10056304.08
      2967572.87     10056969.34      2967734.64     10057458.66
      2967588.99     10057938.91      2968138.04     10058379.94
      2968084.03     10059064.21      2968467.36     10059428.33
      2968548.64     10060089.55       2968362.1     10060704.02
      2968728.76     10061744.76      2969393.13     10062417.62
      2969691.72     10063272.38      2970003.16     10063621.31
      2969933.46     10064108.96      2969279.51      10064548.2
      2970035.19     10064831.55      2970208.77      10065248.7
       2968576.1     10066527.46      2968519.81     10067437.86
      2967588.11     10067468.37      2967670.06     10067808.75
       2968363.6     10068300.84       2968431.6     10068630.56
       2967352.9      10068564.7      2967163.93     10068792.54

Type RM Length L Ch R = 1 ,22276   ,717,717,717
BEGIN DESCRIPTION:
SYCAMORE CREEK 44.0
END DESCRIPTION:
XS GIS Cut Line= 3
      2968521.54     10053527.45      2968807.99      10053792.2
      2969172.59     10054247.95
#Sta/Elev= 30
    4507 1201.05  4522.2  1194.5  4551.8 1181.42  4572.8 1176.66  4649.7 1170.69
  4686.2 1166.85  4749.7 1163.97  4763.8 1161.53  4785.4 1152.24  4863.1 1128.71
  4894.5 1111.91    4912 1110.61  5001.9 1104.03  5004.6 1103.53  5007.9 1104.03
 5015.68 1111.11  5019.3 1115.37  5076.9 1122.18  5104.1 1131.77  5140.9 1136.48
  5147.3 1140.04  5176.2 1143.99  5204.2 1152.89  5211.4 1156.79  5225.8 1159.48
  5232.2 1163.39  5246.6 1165.22  5432.3 1178.26  5452.2 1181.83  5480.7  1184.8
#Mann= 7 ,-1 , 0
    4507     .16       0  4522.2      .1       0  4649.7     .16       0
  5001.9     .07       0  5007.9     .16       0  5204.2      .1       0
  5452.2     .05       0
Bank Sta=4912,5015.68
XS Rating Curve= 0 ,0
Exp/Cntr=0.3,0.1

Type RM Length L Ch R = 1 ,21559   ,579,579,579
BEGIN DESCRIPTION:
SYCAMORE CREEK 43.0
END DESCRIPTION:
XS GIS Cut Line= 3
      2968261.13      10053766.2      2968595.32     10054647.24
      2968742.88     10054833.86
#Sta/Elev= 30
  4291.3 1174.47  4441.3 1165.17  4466.1 1155.67  4502.6 1145.46    4576  1129.8
  4751.5 1112.76  4801.1 1103.33  4806.4 1105.41  4823.4 1101.74  4861.3 1098.05
  4866.7 1100.13  4886.1 1098.02  4891.5  1100.9  4916.3 1097.58  4921.6 1099.16
  4976.5 1097.86  4998.3 1094.14  5001.1 1093.64  5004.3 1094.14  5026.1 1094.73
  5031.5 1096.21 5032.84 1098.92  5056.3 1120.66  5086.4 1164.16  5171.5 1166.79
  5318.4 1181.52  5375.7 1193.05  5396.5 1200.76  5425.4 1208.03  5471.5 1215.49
#Mann= 3 ,-1 , 0
  4291.3     .16       0  4998.3     .07       0  5004.3     .16       0
#XS Ineff= 2 ,-1
  4291.3 4836.48 1102.24 4840.36 4891.48 1100.91
Permanent Ineff=
       T       T
Bank Sta=4976.5,5032.84
XS Rating Curve= 0 ,0
Exp/Cntr=0.3,0.1

Type RM Length L Ch R = 1 ,20980   ,763,763,763
BEGIN DESCRIPTION:
SYCAMORE CREEK 41.0
END DESCRIPTION:
XS GIS Cut Line= 4
      2967905.21     10053766.18      2967861.81     10054195.85
      2968187.33     10054616.86      2968684.07     10054988.33
#Sta/Elev= 30
  4358.4 1175.22  4446.4 1172.98  4496.6 1168.54  4790.3 1161.29  4836.9 1156.03
    4922 1136.06  4942.8 1112.21  4971.8 1097.08 4982.39 1087.83  4992.6  1080.8
  4997.8 1080.02  5000.6 1079.52  5003.8 1080.02  5042.4  1088.2  5100.4 1096.01
  5299.6 1099.66  5427.9 1108.47  5477.9 1124.02  5571.7 1162.79  5735.9 1173.84
    5828 1186.02  5842.6  1193.2  5848.9 1192.77  5871.8 1200.64    5878 1198.11
  5892.6 1205.25  5913.5 1205.06  5921.8 1207.91  5928.1 1206.19  5942.7 1209.16
#Mann= 3 ,-1 , 0
  4358.4     .16       0  4997.8     .07       0  5003.8     .16       0
Bank Sta=4982.39,5042.4
XS Rating Curve= 0 ,0
Exp/Cntr=0.3,0.1

Type RM Length L Ch R = 1 ,20217   ,288,288,288
BEGIN DESCRIPTION:
SYCAMORE CREEK 40.0
END DESCRIPTION:
XS GIS Cut Line= 4
      2967705.57     10054443.29      2967770.67     10054816.51
      2968100.53     10055163.73      2968564.16     10055263.39
#Sta/Elev= 30
  4349.1 1146.42  4491.7  1137.5  4522.1 1131.85  4613.5 1125.25  4674.4 1115.15
  4694.7 1108.14    4728 1102.48  4759.8 1090.91  4844.8 1084.47  4936.6 1080.56
 4955.45 1075.17  4990.2 1069.36    4993 1068.86  4996.2 1069.36  5021.5 1072.17
  5028.4  1075.6  5056.7 1086.13  5078.2 1084.07  5155.8 1097.85  5198.3 1109.85
  5203.4 1113.03  5225.2 1114.85  5279.9 1130.61  5368.4 1148.92  5378.6 1154.87
  5399.1 1163.11  5409.3 1163.98    5440 1162.46  5532.1 1166.26  5681.1 1178.36
#Mann= 4 ,-1 , 0
  4349.1     .16       0  4990.2     .07       0  4996.2     .16       0
  5378.6      .1       0
Bank Sta=4955.45,5028.4
XS Rating Curve= 0 ,0
Exp/Cntr=0.3,0.1

Type RM Length L Ch R = 1 ,19929   ,336,336,336
BEGIN DESCRIPTION:
SYCAMORE CREEK 39.0
END DESCRIPTION:
XS GIS Cut Line= 3
      2967610.07     10054586.45      2967683.86     10055211.47
       2968369.6     10055402.44
#Sta/Elev= 30
  4254.4 1132.46  4352.4 1129.75  4422.8 1125.16  4473.2 1117.13  4493.3 1115.75
  4523.5 1111.12  4573.9 1099.96  4626.9  1092.3  4875.7 1081.92  4961.2 1080.78
  4971.6 1079.78  4987.5 1070.36  4992.3 1065.13  4999.7 1064.05  5002.5 1063.55
  5005.7 1064.05  5020.5 1067.21  5085.8 1070.21  5099.3 1071.25  5127.3 1077.29
  5167.7 1096.94  5179.2 1103.93  5207.1 1114.23  5246.5 1124.62  5251.9 1127.47
  5285.9 1136.78  5320.1 1148.81  5345.3 1154.61  5386.8 1158.79  5595.6 1165.65
#Mann= 3 ,-1 , 0
  4254.4     .16       0  4999.7     .07       0  5005.7     .16       0
Bank Sta=4987.5,5085.8
XS Rating Curve= 0 ,0
Exp/Cntr=0.3,0.1

Type RM Length L Ch R = 1 ,19593   ,531,531,531
BEGIN DESCRIPTION:
SYCAMORE CREEK 38.0
END DESCRIPTION:
XS GIS Cut Line= 4
      2966768.04     10055636.82      2967440.81     10055567.38
      2967926.92     10055571.72      2968282.84     10055636.83
#Sta/Elev= 30
  4028.4 1155.21    4063 1154.29    4120 1152.75  4159.5 1146.91  4179.6  1141.3
  4239.9 1133.94  4270.1 1127.31  4456.9 1108.39  4521.4 1101.28  4551.6 1094.29
  4590.5 1089.28  4595.5 1090.32  4662.2 1084.35  4689.4 1079.97  4842.4 1070.35
    4857 1067.44  4902.4 1063.17  4962.4 1063.27  4999.4    1059  5002.2  1058.5
  5005.4    1059 5016.36 1066.43  5022.4 1071.85  5032.4 1074.73  5092.4 1084.69
  5228.9 1133.65  5282.1 1150.72  5294.1 1152.94  5375.4  1157.8  5552.7 1159.43
#Mann= 6 ,-1 , 0
  4028.4      .1       0    4063     .16       0    4120      .1       0
  4456.9     .16       0  4999.4     .07       0  5005.4     .16       0
Bank Sta=4857,5016.36
XS Rating Curve= 0 ,0
Exp/Cntr=0.3,0.1

Type RM Length L Ch R = 1 ,19062   ,639,639,639
BEGIN DESCRIPTION:
SYCAMORE CREEK 37.0
END DESCRIPTION:
XS GIS Cut Line= 3
      2966794.15      10055892.9      2967809.73     10056049.15
      2968191.67     10055949.32
#Sta/Elev= 30
  4278.1 1154.86  4317.2  1154.6  4363.4  1152.9  4403.9 1146.29  4443.6 1136.02
  4580.2 1113.78  4672.2 1090.67  4788.4 1078.08  4939.3 1069.14  4960.4 1068.29
  4974.8 1064.46 4979.09 1059.67  4990.7 1051.28  4997.8 1051.02  5000.6 1050.52
  5003.8 1051.02  5031.2 1057.27  5162.7 1059.63  5203.2 1062.02  5232.8 1067.92
  5237.9 1066.52  5253.8 1075.47  5301.1 1093.18  5308.4 1093.18  5343.7 1108.36
  5366.3 1110.85  5424.6 1124.17  5586.3 1144.81  5655.7 1151.09  5700.4 1151.74
#Mann= 6 ,-1 , 0
  4278.1      .1       0  4317.2     .16       0  4672.2      .1       0
  4939.3     .16       0  4997.8     .07       0  5003.8     .16       0
#XS Ineff= 2 , 0
                          5169.6         1060.07
Permanent Ineff=
       T       T
Bank Sta=4979.09,5162.7
XS Rating Curve= 0 ,0
Exp/Cntr=0.3,0.1

Type RM Length L Ch R = 1 ,18423   ,417,417,417
BEGIN DESCRIPTION:
SYCAMORE CREEK 36.0
END DESCRIPTION:
XS GIS Cut Line= 4
       2966768.1     10056170.69      2967462.51     10056439.77
      2967883.52     10056448.45      2968204.09     10056023.91
#Sta/Elev= 30
  4008.2 1153.49  4040.8 1152.96  4057.5 1149.67  4087.4 1147.68  4166.5 1128.41
  4226.3 1121.24    4317  1103.8  4359.9 1096.05  4444.3 1085.03  4673.5 1068.45
  4815.5 1063.08  4878.9 1060.67  4928.9 1055.06  4968.9    1053  4978.9 1050.08
  4995.9 1042.98  4998.7 1042.48  5001.9 1042.98  5015.7 1044.46  5048.9 1046.88
 5060.57 1050.51  5088.9 1073.39  5098.9 1078.16  5294.5 1092.24  5352.8 1105.18
  5473.5 1117.64  5488.1 1121.29  5573.4 1128.84  5594.3 1133.61    5706 1148.22
#Mann= 6 ,-1 , 0
  4008.2      .1       0    4317     .16       0  4815.5      .1       0
  4995.9     .07       0  5001.9      .1       0  5015.7     .16       0
Bank Sta=4978.9,5060.57
XS Rating Curve= 0 ,0
Exp/Cntr=0.3,0.1

Type RM Length L Ch R = 1 ,18006   ,420,420,420
BEGIN DESCRIPTION:
SYCAMORE CREEK 35.0
END DESCRIPTION:
XS GIS Cut Line= 4
      2966698.66     10056409.41      2967471.19     10056778.31
      2967900.88     10056964.95      2968382.63     10057095.15
#Sta/Elev= 30
  3988.3  1146.9  4021.3 1146.15  4043.5 1141.58  4121.1 1135.96  4175.4 1129.11
  4420.3 1110.28  4508.9 1099.54  4608.2 1082.22  4675.2 1075.64  4749.9 1062.49
    4890 1053.22  4916.5 1052.07  4945.4 1046.63  4994.8 1038.16  4997.5 1037.66
  5000.8 1038.16  5021.2 1039.64  5037.7    1047  5044.7 1050.78  5212.1 1055.28
  5272.1 1065.41  5277.6 1063.11    5301 1067.66  5326.6 1077.29  5424.3 1091.98
    5466 1102.76  5560.7 1122.53  5642.1 1133.77  5755.8 1144.23  5811.9 1145.29
#Mann= 8 ,-1 , 0
  3988.3     .16       0  4121.1      .1       0  4175.4     .16       0
    4890      .1       0  4994.8     .07       0  5000.8      .1       0
    5466     .05       0  5642.1     .16       0
#XS Ineff= 3 ,-1
 5068.08  5089.8 1051.37 5120.65 5134.66 1052.73 5167.23 5184.07 1053.87
Permanent Ineff=
       T       T       T
Bank Sta=4945.4,5037.7
XS Rating Curve= 0 ,0
Exp/Cntr=0.3,0.1

Type RM Length L Ch R = 1 ,17586   ,441,441,441
BEGIN DESCRIPTION:
SYCAMORE CREEK 34.0
END DESCRIPTION:
XS GIS Cut Line= 4
      2966624.87     10057320.85      2967462.51     10057307.83
      2967757.65     10057190.64      2968303.96     10057247.01
#Sta/Elev= 30
  3990.2 1122.49  4143.8 1113.02  4233.8 1104.45  4273.8 1099.33  4313.8 1091.14
  4473.9 1078.36  4543.9 1069.52  4713.9 1059.08  4941.9 1051.29  4964.9 1048.55
  4974.2 1044.55  4983.8 1040.45  4992.7  1033.4  4995.5  1032.9  4998.7  1033.4
  5081.8 1041.49  5121.5  1041.1  5186.5 1044.05  5216.7 1050.94  5256.9 1074.65
    5322 1088.64  5357.4 1101.54    5416 1113.94    5421 1113.36    5458 1121.92
  5488.1 1124.98  5514.9 1131.27  5608.8 1138.73  5638.9 1143.23  5694.7 1145.55
#Mann= 3 ,-1 , 0
  3990.2     .16       0  4992.7     .07       0  4998.7     .16       0
Bank Sta=4974.2,5186.5
XS Rating Curve= 0 ,0
Exp/Cntr=0.3,0.1

Type RM Length L Ch R = 1 ,17145   ,488,488,488
BEGIN DESCRIPTION:
SYCAMORE CREEK 33.0
END DESCRIPTION:
XS GIS Cut Line= 4
      2966707.34      10057498.8      2967501.57     10057559.56
      2967879.17     10057728.84      2968300.22     10057659.38
#Sta/Elev= 30
    3998 1122.15  4149.6 1109.33    4290 1090.55  4470.5 1078.29  4500.6  1069.7
  4518.5 1067.46  4711.2 1050.83  4892.8  1040.1  4962.3 1035.75  4996.4 1029.23
  4999.1 1028.73  5002.4 1029.23  5037.4 1040.67  5089.2 1053.38  5106.9 1060.15
  5112.4  1059.1  5130.1 1067.25  5135.6 1066.11  5158.7 1079.69  5164.2 1078.47
  5181.9 1083.93  5187.4 1082.32  5205.1 1087.02  5208.2 1085.08  5217.8 1090.02
  5278.6 1108.49  5339.4 1122.71  5400.2 1130.71  5521.8 1140.77  5635.1 1143.09
#Mann= 3 ,-1 , 0
    3998     .16       0  4996.4     .07       0  5002.4     .16       0
Bank Sta=4892.8,5037.4
XS Rating Curve= 0 ,0
Exp/Cntr=0.3,0.1

Type RM Length L Ch R = 1 ,16657   ,550,550,550
BEGIN DESCRIPTION:
SYCAMORE CREEK 32.0
END DESCRIPTION:
XS GIS Cut Line= 4
      2967041.46     10058510.11      2967549.31     10058175.88
      2968009.38     10057793.94      2968313.23     10057724.49
#Sta/Elev= 30
  4271.3 1104.58  4294.8 1099.68  4382.2 1088.69  4454.5 1081.97  4547.8 1076.47
  4779.8 1058.26  4858.1  1054.8  4873.2 1050.82  4908.4 1046.74  4916.2 1043.43
  4957.9 1041.08  4972.2 1038.09 4975.45 1034.72  4986.5 1025.15  4991.3 1024.14
  4994.1 1023.64  4997.3 1024.14  5021.7 1029.51  5050.3 1032.84  5099.8 1034.65
  5263.9 1040.71  5320.1 1045.48    5385 1060.14  5473.5 1100.09  5479.3 1100.09
    5507 1111.04  5549.3 1121.52  5635.2 1131.17  5726.3 1136.27  5788.9  1137.3
#Mann= 3 ,-1 , 0
  4271.3     .16       0  4991.3     .07       0  4997.3     .16       0
Bank Sta=4975.45,5099.8
XS Rating Curve= 0 ,0
Exp/Cntr=0.3,0.1

Type RM Length L Ch R = 1 ,16107   ,600,600,600
BEGIN DESCRIPTION:
SYCAMORE CREEK 31.0
END DESCRIPTION:
XS GIS Cut Line= 4
      2967249.85     10058688.03      2967905.22      10058436.3
      2968300.18     10058180.22      2968456.43     10057754.88
#Sta/Elev= 30
  4069.4 1101.91  4089.3 1099.88  4179.7 1083.61  4343.7 1072.52  4373.7 1067.15
  4537.7  1055.4  4582.1 1049.97  4834.7  1034.8  4870.2 1030.46  4970.6 1025.46
  4997.9 1019.48  5000.6 1018.98  5003.9 1019.48  5079.3 1025.54  5100.5 1031.08
  5112.3 1032.25  5242.2 1041.45  5270.4 1045.61  5308.7 1056.58  5333.8 1066.29
    5345 1073.47  5400.1  1090.7  5408.9 1090.95  5430.6 1099.87  5450.4 1103.97
  5462.1 1108.26  5486.2 1111.93  5516.7 1120.02    5637 1134.61  5695.3 1136.34
#Mann= 6 ,-1 , 0
  4069.4     .16       0  4870.2      .1       0  4997.9     .07       0
  5003.9      .1       0  5112.3     .16       0    5637      .1       0
Bank Sta=4970.6,5079.3
XS Rating Curve= 0 ,0
Exp/Cntr=0.3,0.1

Type RM Length L Ch R = 1 ,15507   ,589,589,589
BEGIN DESCRIPTION:
SYCAMORE CREEK 30.0
END DESCRIPTION:
XS GIS Cut Line= 4
      2967205.54     10058951.62      2967883.08     10058890.68
      2968291.77     10058876.34      2968495.89     10058127.89
#Sta/Elev= 30
  4117.1 1118.57  4135.9 1117.84  4310.8 1104.19  4461.4 1084.51  4531.7  1079.3
  4722.5  1071.3  4732.5 1070.15  4782.7  1054.8  4812.8 1051.22  4831.8 1046.01
  4892.8 1025.18  4922.8 1018.25  4930.7 1016.88  4952.9 1014.18  4999.9 1012.55
  5002.6 1012.05  5005.9 1012.55  5032.9 1016.64  5052.9  1021.6    5123 1027.08
    5296 1030.95  5299.2 1031.12  5555.5 1038.08  5743.8  1040.4  5810.2 1043.24
  5851.7 1048.76  5889.6 1058.58  5924.2 1071.05  5965.7 1080.34  5982.1 1087.92
#Mann= 9 ,-1 , 0
  4117.1      .1       0  4135.9     .16       0  4831.8     .05       0
  4930.7      .1       0  4999.9     .07       0  5005.9      .1       0
    5296     .16       0  5299.2      .1       0  5889.6     .16       0
Bank Sta=4922.8,5032.9
XS Rating Curve= 0 ,0
Exp/Cntr=0.3,0.1

Type RM Length L Ch R = 1 ,14918   ,394,394,394
BEGIN DESCRIPTION:
SYCAMORE CREEK 29.0
END DESCRIPTION:
XS GIS Cut Line= 3
      2967401.72     10059213.21      2968065.81     10059334.74
      2969337.49     10059200.19
#Sta/Elev= 30
    4002  1105.7  4069.9 1101.31  4131.8 1093.45  4273.2 1079.12  4408.9  1072.9
  4517.2 1068.02  4532.5 1063.06  4585.7 1054.86  4876.1 1025.68  4911.1  1021.1
  4931.2 1013.12  4991.5 1009.05  5008.6 1004.54  5011.4 1004.04  5014.6 1004.54
  5092.1  1011.6  5106.2 1010.46  5109.7    1010  5122.2 1009.07  5205.8 1018.27
    5253 1023.26  5283.1 1029.96  5313.3 1045.34  5353.5 1060.27  5399.1 1083.77
  5534.5 1132.56  5604.5 1141.87  5780.3 1149.04  5903.5  1157.7  5955.9  1166.3
#Mann= 11 ,-1 , 0
    4002     .16       0  4131.8      .1       0  4408.9     .16       0
  4876.1      .1       0  5008.6     .07       0  5014.6      .1       0
  5106.2     .05       0  5109.7      .1       0  5205.8     .16       0
  5604.5     .05       0  5903.5      .1       0
#XS Ineff= 2 , 0
                         5096.02         1011.43
Permanent Ineff=
       T       T
Bank Sta=4931.2,5092.1
XS Rating Curve= 0 ,0
Exp/Cntr=0.3,0.1

Type RM Length L Ch R = 1 ,14524   ,415,415,415
BEGIN DESCRIPTION:
SYCAMORE CREEK 28.0
END DESCRIPTION:
XS GIS Cut Line= 3
      2967423.45     10059291.34      2968339.24       10059708.
      2969375.05     10059456.63
#Sta/Elev= 30
  3800.3 1102.94  3941.9 1090.98  4079.4 1076.75    4208 1073.55  4401.1 1065.43
  4420.7 1061.38  4470.3 1056.82    4487 1050.59    4545 1047.54  4614.6 1032.43
  4673.7 1025.26  4921.9 1011.53  4939.4 1008.99  4947.3 1007.94  4974.2 1006.19
  4998.1  999.84  5000.9  999.34  5004.1  999.84  5062.9 1008.86  5289.3 1039.44
  5313.6 1046.19  5350.2 1063.04  5355.4 1061.15    5392 1080.16  5397.1 1077.75
  5412.7 1086.79  5556.8  1134.1  5606.1 1139.85    5768 1144.46  5872.3 1148.99
#Mann= 10 ,-1 , 0
  3800.3     .16       0  3941.9      .1       0    4208     .16       0
  4420.7      .1       0  4614.6     .16       0  4921.9     .05       0
  4947.3     .16       0  4998.1     .07       0  5004.1     .16       0
    5768      .1       0
Bank Sta=4939.4,5062.9
XS Rating Curve= 0 ,0
Exp/Cntr=0.3,0.1

Type RM Length L Ch R = 1 ,14109   ,547,547,547
BEGIN DESCRIPTION:
SYCAMORE CREEK 26.0
END DESCRIPTION:
XS GIS Cut Line= 3
      2967332.34      10060063.9      2968842.72     10060076.93
      2969293.81     10059799.33
#Sta/Elev= 30
  3783.7 1096.57  3879.8 1088.55  3927.3 1081.05  4079.8 1071.55  4220.2 1067.47
  4379.9 1057.83  4419.9 1051.01  4509.9 1048.01  4583.6 1030.97  4619.9 1029.87
  4659.3 1022.26  4839.9 1006.54  4996.9  997.26  4999.6  996.76  5002.9  997.26
  5009.3  998.14  5029.9 1005.99  5209.9 1019.09  5294.1  1036.7  5307.4 1043.88
  5387.5 1057.82  5402.9 1064.53  5445.5 1070.68  5518.9 1089.57  5561.4 1095.67
  5634.8 1102.22  5708.2 1104.53  5714.1 1107.16  5808.8 1109.35  5823.8 1107.27
#Mann= 9 ,-1 , 0
  3783.7     .16       0  3927.3      .1       0  4220.2     .16       0
  4583.6     .05       0  4659.3     .16       0  4996.9     .07       0
  5002.9     .16       0  5009.3      .1       0  5307.4     .16       0
Bank Sta=4839.9,5029.9
XS Rating Curve= 0 ,0
Exp/Cntr=0.3,0.1

Type RM Length L Ch R = 1 ,13562   ,463,463,463
BEGIN DESCRIPTION:
SYCAMORE CREEK 25.0
END DESCRIPTION:
XS GIS Cut Line= 3
      2967267.18     10060259.21      2968781.95     10060693.24
       2969237.7     10060571.71
#Sta/Elev= 30
  3827.6 1100.97  3827.8 1100.97  3922.6 1097.74  4057.9 1082.66  4184.1 1071.59
    4486 1052.78  4585.7 1048.21  4650.7 1034.92  4770.1 1025.51  4810.3 1015.28
  4837.6 1007.69  4931.6  997.01  4954.8  996.04    4991  992.56  4993.8  992.06
    4997  992.56  5027.2  997.34  5094.7 1002.35  5201.1 1001.84  5222.9   998.8
  5267.6 1004.23  5423.2 1022.48  5498.2 1048.85  5538.4 1057.81    5555 1066.65
  5613.4 1080.82  5618.6 1079.53  5653.5 1089.66    5761 1101.22    5875 1109.14
#Mann= 11 ,-1 , 0
  3827.6      .1       0  3827.8     .16       0  4057.9      .1       0
  4184.1     .16       0    4486      .1       0  4810.3     .16       0
  4954.8      .1       0    4991     .07       0    4997      .1       0
  5267.6     .16       0    5761      .1       0
#XS Ineff= 2 , 0
                         5094.47         1002.34
Permanent Ineff=
       T       T
Bank Sta=4931.6,5027.2
XS Rating Curve= 0 ,0
Exp/Cntr=0.3,0.1

Type RM Length L Ch R = 1 ,13099   ,436,436,436
BEGIN DESCRIPTION:
SYCAMORE CREEK 24.0
END DESCRIPTION:
XS GIS Cut Line= 3
      2967123.96     10061118.59       2968938.2     10060923.28
      2969179.98     10060798.07
#Sta/Elev= 30
  3584.4 1113.73  3790.1 1101.23  3858.9  1090.9    3883 1086.73  3956.4 1077.62
  4031.5 1072.11  4061.6 1064.74  4101.9  1065.7  4206.7 1060.54  4242.7  1056.7
  4403.6  1050.1    4474 1037.44  4689.4 1022.93  4799.3 1009.69  4851.8  997.91
  4886.2   986.7    4994  982.04  4996.8  981.54    5000  982.04  5037.2  985.97
  5088.1  994.87  5137.8  999.49  5172.2 1007.06  5218.3 1024.12  5264.2 1046.36
  5288.7 1051.14  5318.9 1064.24  5356.1 1071.46  5489.1 1091.67  5681.4 1095.84
#Mann= 9 ,-1 , 0
  3584.4     .05       0  3858.9     .16       0    3883     .05       0
  4206.7      .1       0  4689.4     .16       0  4851.8      .1       0
    4994     .07       0    5000      .1       0  5088.1     .16       0
Bank Sta=4886.2,5037.2
XS Rating Curve= 0 ,0
Exp/Cntr=0.3,0.1

Type RM Length L Ch R = 1 ,12663   ,602,602,602
BEGIN DESCRIPTION:
SYCAMORE CREEK 23.0
END DESCRIPTION:
XS GIS Cut Line= 4
      2967714.28     10061435.43      2968421.71     10061392.03
      2968790.63     10061322.59      2969114.84     10061032.96
#Sta/Elev= 30
  4086.4 1074.81  4170.7 1068.63  4200.8 1063.36    4283 1056.06  4401.2 1049.86
  4451.3 1037.44  4481.3 1033.97  4631.6 1024.77  4661.7 1021.53  4677.5 1017.68
  4761.9  999.17  4873.3  987.33  4893.6  987.81  4920.1  983.08  4964.8  975.94
  4992.4  975.41  4995.1  974.91  4998.4  975.41  5005.6  975.64  5036.1  984.13
  5196.3 1007.75  5274.8 1029.27  5316.7 1045.01  5359.3 1049.68    5437 1063.71
  5550.7 1065.88  5557.4 1067.56  5564.9 1066.41    5600  1070.2  5605.3 1068.95
#Mann= 5 ,-1 , 0
  4086.4     .05       0    4283      .1       0  4677.5     .16       0
  4992.4     .07       0  4998.4     .16       0
Bank Sta=4920.1,5036.1
XS Rating Curve= 0 ,0
Exp/Cntr=0.3,0.1

Type RM Length L Ch R = 1 ,12061   ,530,530,530
BEGIN DESCRIPTION:
SYCAMORE CREEK 22.0
END DESCRIPTION:
XS GIS Cut Line= 4
      2968230.72     10062294.82      2968729.87     10062047.41
      2969011.99     10061669.81      2969459.06     10061509.21
#Sta/Elev= 30
  4260.8 1064.28  4280.6 1062.96  4325.4 1053.86  4364.4 1047.91  4437.3 1044.16
  4459.7 1034.96  4482.1 1030.26  4540.6 1025.11  4594.2 1021.72  4661.5 1011.53
  4726.9 1006.26  4890.9  987.37 4957.27  976.37    4988  969.51  4990.7  969.01
    4994  969.51  5049.1  974.19  5076.5  975.89  5126.5   979.1  5247.4 1006.65
  5306.8 1017.21  5402.4 1028.41  5470.7 1043.48  5552.7 1048.61  5593.1 1052.61
  5644.4 1056.75  5680.5 1063.16  5734.1 1064.99  5742.4 1068.35  5764.3  1070.3
#Mann= 10 ,-1 , 0
  4260.8      .1       0  4325.4     .05       0  4540.6      .1       0
  4726.9     .05       0    4988    .035       0    4994     .05       0
  5049.1     .16       0  5552.7      .1       0  5593.1     .05       0
  5734.1      .1       0
Bank Sta=4957.27,5076.5
XS Rating Curve= 0 ,0
Exp/Cntr=0.3,0.1

Type RM Length L Ch R = 1 ,11531   ,573,573,573
BEGIN DESCRIPTION:
SYCAMORE CREEK 21.0
END DESCRIPTION:
XS GIS Cut Line= 4
      2968259.42     10062483.17      2968962.51     10062441.51
      2969316.67     10062170.68      2969847.88     10062175.88
#Sta/Elev= 30
  4028.8 1066.79    4128 1063.01  4198.1  1055.1  4228.2  1047.8  4244.6  1048.1
  4298.3 1043.83  4340.5 1030.16  4442.8 1022.09  4498.7  1011.4  4624.5  997.05
  4708.7  988.14  4863.5  984.13  4900.1   981.7    4942  972.02  4964.5   970.4
  4996.9   965.1  4999.6   964.6  5002.9   965.1  5054.4  968.92  5078.8  970.61
  5145.2  977.05  5240.8  987.46  5260.8  987.06  5280.8  981.67  5300.8  984.14
  5440.8 1040.44  5515.1 1051.07  5560.8 1060.12  5695.5 1076.27  5710.2 1078.95
#Mann= 12 ,-1 , 0
  4028.8      .1       0  4244.6     .05       0  4340.5      .1       0
  4624.5     .05       0  4708.7      .1       0  4863.5     .05       0
  4996.9    .035       0  5002.9     .05       0  5054.4      .1       0
  5145.2     .16       0  5515.1      .1       0  5695.5     .16       0
Bank Sta=4964.5,5078.8
XS Rating Curve= 0 ,0
Exp/Cntr=0.3,0.1

Type RM Length L Ch R = 1 ,10958   ,309,309,309
BEGIN DESCRIPTION:
SYCAMORE CREEK 20.0
END DESCRIPTION:
XS GIS Cut Line= 4
      2968269.76      10062686.3       2969144.8     10062795.68
      2969873.97     10062587.34      2970008.71     10062468.14
#Sta/Elev= 30
  3747.1 1063.65  3896.5 1049.72  4009.7 1043.41  4058.2 1031.12  4252.6 1018.67
    4290 1012.13  4360.5 1006.73  4441.2  995.45  4541.3  985.37  4617.2  984.07
  4720.5  980.05  4745.1  979.17  4824.3  974.23  4908.7  967.04  4931.5  965.83
  4993.8  958.47  4996.5  957.97  4999.8  958.47  5032.1  962.37  5048.8  966.37
  5121.6  983.68  5233.7 1026.08  5256.8  1038.2    5288 1047.77  5319.2 1062.85
  5371.2 1076.36    5387 1083.27  5435.3 1092.43  5505.7 1096.88  5567.2  1101.5
#Mann= 13 ,-1 , 0
  3747.1      .1       0  3896.5     .05       0  4009.7      .1       0
  4541.3     .05       0  4617.2      .1       0  4720.5     .16       0
  4745.1      .1       0  4824.3     .05       0  4931.5      .1       0
  4993.8     .07       0  4999.8      .1       0  5032.1     .16       0
  5505.7      .1       0
Bank Sta=4908.7,5048.8
XS Rating Curve= 0 ,0
Exp/Cntr=0.3,0.1

Type RM Length L Ch R = 1 ,10649   ,382,382,382
BEGIN DESCRIPTION:
SYCAMORE CREEK 19.0
END DESCRIPTION:
XS GIS Cut Line= 4
      2968457.27     10063217.55      2969238.55      10063123.8
      2969868.76     10062879.01      2970050.59     10062728.35
#Sta/Elev= 30
  3834.5 1046.11  3855.8  1044.5  3904.9 1032.15    4101 1022.79    4373 1004.68
  4500.5  995.18  4559.3  989.13  4618.8  979.73  4728.8  976.51  4783.9  974.45
  4878.7   971.6  4921.6  965.48  4989.9  956.35  4992.7  955.85  4995.9  956.35
  5017.5  957.42  5052.7   965.4  5107.2  977.93  5131.7  995.36  5137.1  994.43
  5156.2 1008.01  5161.6 1006.66  5186.1 1024.27  5191.5 1023.23  5210.7 1034.13
  5240.6 1046.02  5245.9 1045.39  5270.5 1060.06  5407.5 1090.36  5533.6 1096.51
#Mann= 10 ,-1 , 0
  3834.5     .05       0    4101      .1       0    4373     .05       0
  4500.5     .16       0  4559.3      .1       0  4728.8     .05       0
  4783.9      .1       0  4921.6     .16       0  4989.9     .07       0
  4995.9     .16       0
Bank Sta=4921.6,5052.7
XS Rating Curve= 0 ,0
Exp/Cntr=0.3,0.1

Type RM Length L Ch R = 1 ,10267   ,565,565,565
BEGIN DESCRIPTION:
SYCAMORE CREEK 18.0
END DESCRIPTION:
XS GIS Cut Line= 4
      2968498.92     10063439.77      2969479.87     10063483.18
      2969944.28     10063218.42      2970104.15     10062963.49
#Sta/Elev= 30
  3723.5 1047.74  3753.1 1045.52  3803.1 1034.89  3843.2 1030.09  4073.4 1019.79
  4150.5 1011.53  4155.5 1013.56  4173.5 1010.17  4231.2 1007.52  4307.8 1000.98
  4443.8  992.78  4601.9  975.46  4795.2  968.25  4959.7  959.33  4960.2   959.3
  4994.2  952.91  4996.9  952.41  5000.2  952.91  5049.1  959.12  5164.3 1002.08
  5201.7  1014.5  5233.3 1020.23  5269.1 1035.22  5296.8 1040.78  5312.1  1047.7
  5333.3 1050.72  5348.6 1056.19  5448.8 1070.29  5464.1 1074.78  5540.9 1082.05
#Mann= 7 ,-1 , 0
  3723.5      .1       0  4231.2     .16       0  4307.8     .05       0
  4795.2      .1       0  4960.2     .16       0  4994.2     .07       0
  5000.2     .16       0
Bank Sta=4959.7,5049.1
XS Rating Curve= 0 ,0
Exp/Cntr=0.3,0.1

Type RM Length L Ch R = 1 ,9702    ,429,429,429
BEGIN DESCRIPTION:
SYCAMORE CREEK 17.0
END DESCRIPTION:
XS GIS Cut Line= 4
      2968702.95     10063860.78      2969831.43     10063739.25
      2970426.05     10063856.44      2970777.65     10064142.93
#Sta/Elev= 30
  3698.2 1022.49  3798.3 1019.82  3865.9 1015.43    3915 1011.01  4055.8 1006.06
  4151.9  997.73  4493.9  987.43  4555.8  987.29  4585.6  981.66  4719.6  963.61
  4840.4  963.09  4879.1  958.15  4884.2  960.26  4911.7  955.05  5000.5  948.91
  5003.2  948.41  5006.5  948.91  5033.2  951.32  5105.4  949.33  5283.6  951.34
  5351.4  950.45  5380.2  954.93  5402.7  959.34  5431.5  969.36    5489    1002
  5509.8 1010.04  5689.2 1022.12  5709.4 1023.71    5759 1034.84  5892.8 1040.36
#Mann= 11 ,-1 , 0
  3698.2      .1       0  3798.3     .05       0  3865.9      .1       0
  4151.9     .05       0  4493.9     .16       0  4585.6      .1       0
  5000.5     .07       0  5006.5      .1       0  5283.6     .16       0
  5380.2     .05       0  5689.2      .1       0
Bank Sta=4911.7,5380.2
XS Rating Curve= 0 ,0
Exp/Cntr=0.3,0.1

Type RM Length L Ch R = 1 ,9408    ,110,110,110
BEGIN DESCRIPTION:
Mapping XS b3df0c54
END DESCRIPTION:
XS GIS Cut Line= 4
      2968678.91     10063882.75      2969894.14     10063934.83
      2970081.64     10064155.32      2970362.92     10064245.61
#Sta/Elev= 30
  3659.7  1024.3    3798 1021.87  3899.5  1019.5  3952.9 1014.64  4093.5 1006.66
  4189.7  999.27  4259.8  996.26    4283   991.9  4309.9  986.48  4369.9  967.94
  4409.9  959.85  4497.5  955.66  4502.5  953.96  4560.3  954.67    4856  956.81
  4878.6  957.12  4920.9  950.35  4992.7  948.64  5059.6  948.58  5062.3  948.08
  5065.6  948.58  5076.9   949.5    5112  969.72  5136.7  976.56    5172  987.92
  5204.1  992.34  5372.2  1006.3  5407.3 1008.94  5434.2 1013.25  5460.9 1014.44
#Mann= 12 ,-1 , 0
  3659.7      .1       0    3798     .05       0  3952.9      .1       0
  4093.5     .05       0    4283     .16       0  4560.3     .05       0
    4856      .1       0  4992.7     .16       0  5059.6     .07       0
  5065.6     .16       0  5136.7     .05       0  5372.2      .1       0
Bank Sta=5059.6,5065.6
XS Rating Curve= 0 ,0
Exp/Cntr=0.3,0.1

Type RM Length L Ch R = 1 ,9298    ,43,43,43
BEGIN DESCRIPTION:
Mapping XS 48f367e1
END DESCRIPTION:
XS GIS Cut Line= 5
      2968670.16     10063907.05      2969852.19     10064059.03
      2969895.66     10064060.92      2969957.91     10064215.57
      2970371.59     10064320.26
#Sta/Elev= 30
  3706.7 1026.67  3869.9 1023.89  3925.7 1023.31  4027.6 1019.12  4222.5 1003.29
  4279.7  996.67  4299.8   991.2  4321.5  981.51  4340.2  974.14  4351.3     967
  4380.5  957.79  4455.2  952.64  4618.3  953.16  4733.4  954.26  4763.6  948.39
  4871.5  948.18  4874.3  947.68  4877.5  948.18    4915  949.04  5059.1  948.68
  5085.1  951.69  5093.7  954.05    5099  958.59  5111.6  958.45  5140.2  969.63
  5191.8  978.27  5212.3  984.53    5264  992.33  5410.7 1004.75  5535.4 1015.39
#Mann= 14 ,-1 , 0
  3706.7      .1       0  3869.9     .05       0  3925.7      .1       0
  4222.5     .16       0  4321.5     .05       0  4455.2      .1       0
  4618.3     .05       0  4871.5     .07       0  4877.5     .05       0
    4915     .16       0  5059.1      .1       0  5111.6     .16       0
  5212.3     .05       0  5410.7      .1       0
Bank Sta=4871.5,4877.5
XS Rating Curve= 0 ,0
Exp/Cntr=0.3,0.1

Type RM Length L Ch R = 1 ,9255    ,77,77,77
BEGIN DESCRIPTION:
Mapping XS 28ceafcd
END DESCRIPTION:
XS GIS Cut Line= 5
      2968645.83     10063937.43      2969802.13     10064105.84
      2969871.57     10064111.05      2969914.97     10064249.94
      2970366.23     10064369.23
#Sta/Elev= 30
  3742.9 1028.92  3846.6 1028.99  4048.7 1022.55  4101.6 1020.08  4139.7 1014.04
  4282.7 1004.55  4301.4 1002.73  4331.7  994.58  4381.8  968.43  4412.5  959.19
  4441.8  954.94  4549.2  951.81  4766.2  952.97  4797.1  947.03    4834  943.25
  4836.7  942.75    4840  943.25  4877.3  949.21  4917.7  955.97  5040.1  954.59
  5058.4  953.45  5085.7  955.08  5090.9  953.07  5123.4  954.39  5140.5  956.55
  5171.9  966.14  5272.9  986.01  5314.3  991.99  5455.9 1003.93  5593.3 1016.19
#Mann= 11 ,-1 , 0
  3742.9      .1       0  4282.7     .16       0  4381.8     .05       0
  4549.2      .1       0    4834     .07       0    4840      .1       0
  4877.3     .16       0  5040.1      .1       0  5171.9     .16       0
  5272.9     .05       0  5455.9      .1       0
Bank Sta=4834,4840
XS Rating Curve= 0 ,0
Exp/Cntr=0.3,0.1

Type RM Length L Ch R = 1 ,9178    ,291,291,291
BEGIN DESCRIPTION:
SYCAMORE CREEK 16.0
END DESCRIPTION:
XS GIS Cut Line= 4
      2968641.55     10064016.43      2969799.52     10064137.96
      2969875.91     10064301.15      2970353.38     10064407.06
#Sta/Elev= 30
  3806.9  1044.4  3897.8 1036.55  3922.1  1031.9  4044.1 1026.35  4175.8 1020.64
  4211.6 1014.53  4309.8 1008.73  4345.8 1004.03  4366.9  998.34  4417.2  969.42
  4444.6  960.31  4507.6  953.29  4644.2  951.64  4809.3  952.03  4839.5  943.24
  4896.8  941.42  4899.5  940.92  4902.8  941.42  4938.5  948.63  4971.2  948.04
  5000.2  942.89  5073.2  945.08  5078.7  946.46    5088  954.64    5096  956.67
    5195  955.57  5233.9  968.08    5334     987  5459.4  999.07  5640.5 1014.64
#Mann= 13 ,-1 , 0
  3806.9      .1       0  3897.8     .05       0  4044.1      .1       0
  4345.8     .16       0  4444.6     .05       0  4644.2      .1       0
  4896.8     .07       0  4902.8      .1       0  4938.5     .16       0
  5000.2      .1       0  5233.9     .16       0    5334     .05       0
  5459.4      .1       0
Bank Sta=4896.8,4902.8
XS Rating Curve= 0 ,0
Exp/Cntr=0.3,0.1

Type RM Length L Ch R = 1 ,8887    ,400,400,400
BEGIN DESCRIPTION:
SYCAMORE CREEK 15.0
END DESCRIPTION:
XS GIS Cut Line= 4
      2968629.41     10064264.69      2969520.01     10064186.57
      2969598.13     10064384.49      2970329.08     10064455.67
#Sta/Elev= 30
  3993.1  1057.1  4022.3 1049.06  4048.6 1050.03  4142.7 1046.01  4192.9 1033.39
  4363.6 1022.29  4401.7 1016.37    4484 1009.54  4513.8 1003.33  4519.1    1003
  4554.3  982.18  4584.4  968.04  4636.6  956.17  4714.9  950.63  4898.4  949.98
  4956.7     940  4978.7  937.12  4998.2  936.12    5001  935.62  5004.2  936.12
  5096.8  948.46  5168.5  950.66  5258.2  955.28  5348.2  958.47  5381.6  955.45
  5455.6  968.98    5482  975.79  5554.4  986.44  5653.1  996.88  5834.3 1013.99
#Mann= 13 ,-1 , 0
  3993.1      .1       0  4048.6     .05       0  4513.8      .1       0
  4636.6     .05       0  4956.7      .1       0  4978.7     .05       0
  4998.2    .035       0  5004.2     .05       0  5168.5      .1       0
  5258.2     .05       0  5455.6      .1       0  5554.4     .16       0
  5653.1      .1       0
Bank Sta=4998.2,5004.2
XS Rating Curve= 0 ,0
Exp/Cntr=0.3,0.1

Type RM Length L Ch R = 1 ,8487    ,725,725,725
BEGIN DESCRIPTION:
SYCAMORE CREEK 14.0
END DESCRIPTION:
XS GIS Cut Line= 4
      2968645.82     10064560.29      2969697.92     10064515.15
      2970284.73     10064501.26      2970590.26     10064438.76
#Sta/Elev= 30
  4370.6 1054.81  4393.3 1050.15  4478.8 1047.99  4553.4 1031.69  4673.5 1023.36
  4701.7  1018.9  4753.6 1010.96    4810 1008.32  4876.1 1003.48  4923.8  993.01
  4943.8  981.32  4953.8  971.08  4965.5  952.09  4973.8  941.63  4983.8  935.42
  5000.8   932.5  5003.6     932  5006.8   932.5  5107.8  941.68    5134  946.84
  5179.9  949.09  5476.6  951.72  5575.4  955.79  5624.3  957.91  5764.3  985.46
  5791.3  988.82  6021.4  1011.9  6218.2 1022.34    6290 1035.79  6322.5 1037.51
#Mann= 11 ,-1 , 0
  4370.6     .05       0  4478.8      .1       0  4701.7     .05       0
    4810      .1       0  4965.5     .16       0  5000.8     .07       0
  5006.8     .16       0  5179.9      .1       0  5476.6     .05       0
  5575.4     .16       0  5791.3      .1       0
Bank Sta=4973.8,5107.8
XS Rating Curve= 0 ,0
Exp/Cntr=0.3,0.1

Type RM Length L Ch R = 1 ,7762    ,427,427,427
BEGIN DESCRIPTION:
SYCAMORE CREEK 13.0
END DESCRIPTION:
XS GIS Cut Line= 4
      2968704.91     10065101.95      2969753.48     10064994.31
      2969965.28     10064664.45      2970814.71     10064432.16
#Sta/Elev= 30
  3676.1 1049.36  3683.5 1049.32  3710.7 1047.75  3760.1 1040.12  3790.3 1030.77
  3951.1 1019.47  3981.3 1012.96  4098.1   998.4  4354.4  971.68  4433.6  964.11
    4490  954.88  4604.5  951.35  4674.9  937.24  4957.4  932.98  5002.8  926.27
  5030.1  932.11  5039.4  940.61  5051.7   943.8  5081.6  948.24  5111.2  947.55
  5128.9  951.16    5177  964.02  5229.2  983.12  5280.3  992.51  5457.2 1011.65
  5664.6 1022.37  5751.6 1035.54  5944.8 1036.58  5974.2 1043.46  6002.8 1045.14
#Mann= 8 ,-1 , 0
  3676.1     .16       0  3683.5     .05       0  3710.7      .1       0
  4354.4     .16       0  4957.4     .07       0  5030.1      .1       0
  5128.9     .16       0  5280.3      .1       0
#XS Ineff= 2 , 0
         4849.58  935.32
Permanent Ineff=
       T       T
Bank Sta=4957.4,5030.1
XS Rating Curve= 0 ,0
Exp/Cntr=0.3,0.1

Type RM Length L Ch R = 1 ,7335    ,538,538,538
BEGIN DESCRIPTION:
SYCAMORE CREEK 12.0
END DESCRIPTION:
XS GIS Cut Line= 4
      2968799.32     10065139.43      2969931.26     10065066.51
      2970514.59     10065101.23      2971080.59     10065767.93
#Sta/Elev= 30
  3645.9 1045.93    3683 1034.81  3705.2 1030.19  3805.4  1023.6  3875.5 1011.88
    4054  991.25  4122.2  979.58  4336.5  958.66  4366.5  949.84  4396.6  946.25
  4496.8  944.51    4586  940.47  4627.1  936.03  4847.5  934.57  4947.7  931.44
  4967.7  927.62  4997.5     923  5057.9  929.61    5128  924.89  5198.1   932.4
  5317.9  944.92  5454.3  952.61    5596  957.71  5617.1  962.05  5723.4  971.43
  5794.8  983.28  6003.4  999.99  6091.5 1006.18  6141.9 1012.96  6239.1 1016.63
#Mann= 9 ,-1 , 0
  3645.9     .05       0    3683      .1       0    4054     .16       0
  4967.7     .05       0  4967.7     .07       0    5128      .1       0
  5454.3      .1       0  6003.4     .05       0  6091.5      .1       0
Bank Sta=4947.7,5198.1
XS Rating Curve= 0 ,0
Exp/Cntr=0.3,0.1

Type RM Length L Ch R = 1 ,6797    ,550,550,550
BEGIN DESCRIPTION:
SYCAMORE CREEK 11.0
END DESCRIPTION:
XS GIS Cut Line= 4
       2968719.4     10065236.64      2969872.23     10065316.51
      2970129.17     10065684.56      2970545.87     10065889.44
#Sta/Elev= 30
  3610.6 1053.73  3723.3 1045.72    3770 1031.46  3834.6 1026.32  3890.3 1021.02
  3920.5 1013.92  3986.1  1004.9    4181  976.02  4217.8  965.05  4251.2  961.66
  4281.3  949.31    4315   944.4  4413.6   938.5  4478.7  937.99  4789.6  940.48
    4855  938.64  4905.6  931.38    4995  920.66  4997.8  920.16    5001  920.66
  5051.6  922.87  5063.5  923.98 5073.86  930.86  5084.4  935.53  5092.1  949.78
  5099.2  956.64  5334.6  969.37  5435.5  984.64  5561.8  990.08  5679.4  994.67
#Mann= 13 ,-1 , 0
  3610.6     .16       0  3723.3      .1       0  3834.6     .05       0
  3920.5      .1       0  3986.1     .16       0    4315      .1       0
  4413.6     .05       0  4478.7      .1       0    4995     .07       0
    5001      .1       0  5051.6     .16       0  5435.5      .1       0
  5561.8     .16       0
#XS Ineff= 2 , 0
         4789.77  941.55
Permanent Ineff=
       T       T
Bank Sta=4905.6,5073.86
XS Rating Curve= 0 ,0
Exp/Cntr=0.3,0.1

Type RM Length L Ch R = 1 ,6247    ,682,682,682
BEGIN DESCRIPTION:
SYCAMORE CREEK 10.0
END DESCRIPTION:
XS GIS Cut Line= 4
      2968493.78     10065479.71      2969410.42     10065587.34
      2969674.31     10065958.87      2970413.69     10065969.28
#Sta/Elev= 30
  3864.9 1072.38  3995.9 1062.49  4050.9 1053.85  4161.6 1044.79    4212 1030.12
  4286.4 1027.04  4391.3 1012.29  4457.7 1002.71  4534.2  966.92  4554.3  952.66
    4589  941.52  4634.8  935.56  4755.7   933.2  4927.9  932.49  4955.1  923.14
  4969.7  918.15  4996.2  916.85  4998.9  916.35  5002.2  916.85  5035.5  918.76
  5100.1  917.32  5150.5  923.85  5176.9  927.62  5192.3  929.01  5297.7  939.12
  5377.7  956.69  5443.7  962.99  5738.7  976.25  5867.8  985.25    5983  986.67
#Mann= 12 ,-1 , 0
  3864.9      .1       0  3995.9     .05       0  4391.3     .16       0
    4589     .05       0  4755.7      .1       0  4996.2     .07       0
  5002.2      .1       0  5035.5     .16       0  5176.9      .1       0
  5192.3     .16       0  5443.7      .1       0  5738.7     .16       0
Bank Sta=4955.1,5150.5
XS Rating Curve= 0 ,0
Exp/Cntr=0.3,0.1

Type RM Length L Ch R = 1 ,5565    ,501,501,501
BEGIN DESCRIPTION:
SYCAMORE CREEK 9.0
END DESCRIPTION:
XS GIS Cut Line= 4
      2968393.05     10065535.25      2968900.01     10066021.37
      2969406.95     10066677.62      2969879.18     10066868.59
#Sta/Elev= 30
    4073 1078.11  4238.4 1066.32  4304.4 1057.58    4401 1044.43  4493.1 1012.43
  4549.7   985.4  4556.7  979.27  4570.8   972.7  4653.1  948.18  4690.9  938.39
  4733.4  932.25  4861.7  926.04  4917.8  919.56  4940.5  911.32  5001.8  909.45
  5004.5  908.95  5007.8  909.45  5125.2  920.33  5125.4  920.37  5154.2  925.67
  5230.5  929.57  5382.4  937.51    5482  945.46  5567.2  962.81  5627.8  966.06
  5703.3  976.03  5767.3  980.27  5824.2  988.37  6037.9  999.54    6114 1002.26
#Mann= 10 ,-1 , 0
    4073      .1       0  4304.4     .16       0  4653.1      .1       0
  5001.8     .07       0  5007.8      .1       0  5125.4     .05       0
  5230.5      .1       0  5382.4     .16       0  5767.3     .05       0
  6037.9     .16       0
Bank Sta=4917.8,5125.2
XS Rating Curve= 0 ,0
Exp/Cntr=0.3,0.1

Type RM Length L Ch R = 1 ,5064    ,565,565,565
BEGIN DESCRIPTION:
SYCAMORE CREEK 8.0
END DESCRIPTION:
XS GIS Cut Line= 4
      2968090.97     10065486.63      2968264.59     10066059.56
      2969011.12      10066917.2      2969493.63      10067111.6
#Sta/Elev= 30
  3854.6 1087.65  3931.7 1077.54  3975.2 1075.57  4043.4 1071.78    4210 1061.69
  4251.6 1054.43  4346.9 1045.66  4459.3 1023.91  4510.3  998.69  4558.2  964.26
  4607.6  939.59    4636  930.49  4867.9  924.32  4912.3   917.4  4940.2  912.77
  4994.8  906.72  4997.5  906.22  5000.8  906.72  5083.5  915.65  5089.9  917.98
  5104.1  922.74    5125  924.28  5288.3  924.21  5442.1  928.86    5501  932.46
  5529.5   942.8  5550.4  955.98  5564.6  961.13  5778.9  970.36  6110.5  992.59
#Mann= 12 ,-1 , 0
  3854.6      .1       0  3931.7     .16       0  3975.2      .1       0
  4043.4     .16       0  4251.6      .1       0  4510.3     .05       0
  4867.9      .1       0  4940.2     .16       0  4994.8     .07       0
  5000.8     .16       0  5083.5      .1       0  5442.1     .16       0
#XS Ineff= 2 , 0
                          5123.7          924.47
Permanent Ineff=
       T       T
Bank Sta=4912.3,5089.9
XS Rating Curve= 0 ,0
Exp/Cntr=0.3,0.1

Type RM Length L Ch R = 1 ,4499    ,367,367,367
BEGIN DESCRIPTION:
SYCAMORE CREEK 7.0
END DESCRIPTION:
XS GIS Cut Line= 2
      2967459.07     10066517.91      2969444.34     10067284.95
#Sta/Elev= 30
  3761.6 1050.93  3765.1 1048.18  3789.7 1046.38  3825.3 1038.33  3967.7 1023.35
  4061.1 1001.93  4157.7  974.76    4248   958.1  4286.5  953.14  4680.5  932.89
    4793  926.14    4833  915.48  4840.3  914.52  4877.5   913.7  4896.7  907.03
    4959  902.98  4961.8  902.48    4965  902.98  5048.4   906.3  5090.3  915.65
    5184  919.35  5221.5  921.86  5283.3  929.31  5319.2  942.81  5326.1  947.25
  5336.9  960.56  5349.2  964.96  5458.3  972.78  5690.6  980.41  5889.9  993.84
#Mann= 11 ,-1 , 0
  3761.6     .16       0  3967.7      .1       0    4248     .05       0
  4286.5      .1       0  4680.5     .05       0  4840.3      .1       0
    4959     .07       0    4965      .1       0  5048.4     .16       0
    5184      .1       0  5221.5     .16       0
#XS Ineff= 2 , 0
                         5122.16          918.82
Permanent Ineff=
       T       T
Bank Sta=4833,5090.3
XS Rating Curve= 0 ,0
Exp/Cntr=0.3,0.1

Type RM Length L Ch R = 1 ,4132    ,1149,1149,1149
BEGIN DESCRIPTION:
SYCAMORE CREEK 6.0
END DESCRIPTION:
XS GIS Cut Line= 3
       2967403.5     10066549.16      2968747.23     10067413.73
      2969423.88      10067417.2
#Sta/Elev= 30
    3574 1041.39  3588.8 1041.69  3594.7 1038.83  3615.9 1036.28  3718.9 1031.36
  3770.2 1025.83    3879 1001.11  3948.7  982.09  4021.3  965.23  4093.9  952.59
  4187.7  940.73  4491.3  928.95  4717.3  920.09  4759.5  914.18  4889.6  909.51
  4947.4  902.13  4971.2     902  4998.3  898.68  5001.6  899.18  5034.9  903.02
 5045.45  914.02    5056  922.17  5107.5  945.58  5122.7  956.06  5143.9  963.49
  5433.1  969.61  5593.1  979.43  5693.1  988.92  5773.1  991.42  5848.5  997.73
#Mann= 5 ,-1 , 0
    3574     .16       0    3879      .1       0  4491.3     .16       0
  4889.6     .05       0  5001.6     .16       0
Bank Sta=4759.5,5045.45
XS Rating Curve= 0 ,0
Exp/Cntr=0.3,0.1

Type RM Length L Ch R = 1 ,2983    ,995,995,995
BEGIN DESCRIPTION:
SYCAMORE CREEK 5.0
END DESCRIPTION:
XS GIS Cut Line= 4
       2967122.2     10067462.34      2967698.62     10067528.31
       2968188.2     10067708.87       2969493.6     10067469.32
#Sta/Elev= 30
  4536.2 1035.96    4774 1023.97  4784.1 1020.55  4852.9  975.29  4857.9  976.05
  4884.7  951.23  4942.1  923.14    4971  898.34  4992.4  890.76  4995.2  890.26
  5025.6  895.69  5065.9  892.61  5144.7  895.01  5180.4   897.4    5200  898.38
  5402.6  907.53  5438.4  918.07  5524.4  925.22  5800.6  925.35  5943.5  932.14
  6081.5  926.55  6134.6  930.34    6251  949.26    6299  945.57  6304.1  948.53
  6350.2  941.16  6421.3  963.38  6512.8  968.57  6716.2   988.9  6965.4 1000.17
#Mann= 4 ,-1 , 0
  4536.2      .1       0  4992.4     .05       0  5144.7      .1       0
    5200     .16       0
Bank Sta=4971,5180.4
XS Rating Curve= 0 ,0
Exp/Cntr=0.3,0.1

Type RM Length L Ch R = 1 ,1988    ,452,452,452
BEGIN DESCRIPTION:
SYCAMORE CREEK 4.0
END DESCRIPTION:
XS GIS Cut Line= 4
      2967233.37     10067830.41      2968045.84      10068267.9
       2968500.7     10068076.93      2969323.59     10068194.98
#Sta/Elev= 30
  3889.3 1013.08  4147.6  979.28  4183.9   975.2  4360.7   964.8  4456.3  952.29
  4510.1  938.58  4598.2  924.46  4603.9  928.89  4620.1  921.26  4625.8  925.13
    4642  919.58  4647.7  924.19  4663.9  919.19  4669.6  923.81  4702.9  918.65
  4729.7  923.91  4745.9  918.76  4751.6  922.99  4795.4  922.35  4884.6  894.27
  4996.3  883.51    4999  883.01  5002.3  883.51  5075.2  894.16  5112.4  900.69
  5388.8  924.73  5459.3  935.77  5565.8  965.38  5741.6  990.74  6136.7  995.54
#Mann= 9 ,-1 , 0
  3889.3     .16       0  4147.6      .1       0  4183.9     .16       0
  4510.1     .05       0  4702.9     .16       0  4884.6     .05       0
  4996.3    .035       0  5002.3     .05       0  5112.4     .16       0
Bank Sta=4884.6,5075.2
XS Rating Curve= 0 ,0
Exp/Cntr=0.3,0.1

Type RM Length L Ch R = 1 ,1536    ,799,799,799
BEGIN DESCRIPTION:
SYCAMORE CREEK 3.0
END DESCRIPTION:
XS GIS Cut Line= 4
       2967389.6     10067979.71       2968188.2     10068472.76
       2968375.7     10068549.15      2968833.78     10068583.85
#Sta/Elev= 30
  3789.1   982.7  3973.8  965.55  4000.9  960.28  4010.4   961.2    4105  954.23
  4211.4  934.71  4263.4  930.05  4437.2  921.52  4583.9  919.06    4721  906.81
  4850.8  906.23    4934  900.68    4963   891.1    4983  881.55  5000.1  879.95
  5002.8  879.45  5006.1  879.95  5033.2  880.19  5123.4  890.74  5153.5  901.67
    5189  924.23  5213.7  935.38  5223.7  944.83  5233.7  960.29  5243.8  969.89
  5263.8   986.5  5273.9  991.53    5314  995.02    5334  999.38  5389.5 1001.77
#Mann= 3 ,-1 , 0
  3789.1     .16       0  5000.1     .07       0  5006.1     .16       0
Bank Sta=4963,5123.4
XS Rating Curve= 0 ,0
Exp/Cntr=0.3,0.1

Type RM Length L Ch R = 1 ,737     ,499,499,499
BEGIN DESCRIPTION:
SYCAMORE CREEK 2.0
END DESCRIPTION:
XS GIS Cut Line= 4
       2967285.4     10067983.16      2967722.92     10068285.26
      2967778.48     10068674.15      2968328.74     10068909.48
#Sta/Elev= 30
  4206.4   993.4    4273  983.27  4446.1  966.96  4574.7  936.63  4619.1  937.63
  4669.8  933.46  4837.6  913.44  4953.9  884.35    4958  884.17  4996.2  875.71
  4998.9  875.21  5002.2  875.71  5024.6  879.76  5100.4  879.25  5120.4   886.5
  5128.2  890.49  5163.1  888.85  5168.5  893.54  5192.1  893.54  5197.5  896.65
  5215.7  897.01  5250.5  905.24  5291.9  907.64  5320.9   914.5  5344.5   912.7
  5435.4  925.97  5467.9  923.23    5526  931.02  5678.4  939.53  5729.4  949.22
#Mann= 4 ,-1 , 0
  4206.4     .16       0    4958      .1       0  4996.2     .07       0
  5002.2      .1       0
#XS Ineff= 1 ,-1
 5133.64 5180.91  891.19
Permanent Ineff=
       T
Bank Sta=4953.9,5120.4
XS Rating Curve= 0 ,0
Exp/Cntr=0.3,0.1
