HEC-RAS study YEAGER CREEK.prj: YEAGER CREEK Base Level Engineering

--- YEAGER CREEK.g01 (geometry) --- (continued)

Type RM Length L Ch R = 1 ,20574   ,597,597,597
BEGIN DESCRIPTION:
YEAGER CREEK 35.0
END DESCRIPTION:
XS GIS Cut Line= 4
      2943485.74     10043331.68      2943978.79     10043880.28
      2944673.23     10044123.34      2945933.58     10044237.91
#Sta/Elev= 30
  3986.4 1223.92  4258.5 1212.93  4343.7 1202.42    4358 1199.65  4365.4 1194.69
  4372.2 1193.47  4386.4  1180.6  4400.6 1174.11  4471.6 1154.89  4641.2 1147.69
    4837  1143.5    4874 1135.01    4925 1127.72  4961.8 1129.55  4996.1 1125.18
  4998.9 1124.68  5002.1 1125.18  5018.5 1129.56  5094.5  1135.8  5202.2 1139.28
    5455 1138.54  5652.5 1145.77  5796.4  1149.3  5821.9 1151.77  5876.7 1155.43
  5926.9 1162.71  6183.5 1181.08  6309.7 1192.52  6348.6  1195.8  6725.3 1207.74
#Mann= 10 ,-1 , 0
  3986.4     .16       0    4837      .1       0  4996.1     .07       0
  5002.1      .1       0  5202.2     .05       0    5455      .1       0
  5652.5     .16       0  5821.9      .1       0  6183.5     .05       0
  6309.7      .1       0
#XS Ineff= 2 , 0
                         5274.33         1140.35
Permanent Ineff=
       T       T
Bank Sta=4874,5094.5
XS Rating Curve= 0 ,0
Exp/Cntr=0.3,0.1

Type RM Length L Ch R = 1 ,19977   ,1498,1498,1498
BEGIN DESCRIPTION:
YEAGER CREEK 34.0
END DESCRIPTION:
XS GIS Cut Line= 4
      2943100.35      10044178.9      2943829.48     10044362.92
      2944405.87     10044779.59      2945734.61     10045025.91
#Sta/Elev= 30
  4019.3 1238.45    4031 1238.09  4120.5 1233.87  4151.4 1229.36  4261.8 1225.64
  4460.8 1211.51  4522.7 1204.34  4584.6 1186.22  4625.9 1165.23  4636.5 1156.79
  4687.7 1138.97  4718.7 1135.79  4914.9    1131  4997.7 1119.15  5000.5 1118.65
  5003.7 1119.15  5042.5 1131.33  5122.2 1150.03  5173.1 1152.72    5330 1156.47
  5424.5 1154.67  5589.8 1155.15  5911.6 1164.63  6034.4  1165.6  6283.8 1175.38
  6614.1 1191.41  6646.6 1195.83  6746.9 1200.42  6821.1 1202.77  6833.9 1202.97
#Mann= 12 ,-1 , 0
  4019.3      .1       0    4031     .16       0  4997.7     .07       0
  5003.7     .16       0  5173.1      .1       0    5330     .16       0
  5424.5      .1       0  5911.6     .16       0  6283.8      .1       0
  6646.6     .16       0  6746.9      .1       0  6821.1     .16       0
Bank Sta=4914.9,5042.5
XS Rating Curve= 0 ,0
Exp/Cntr=0.3,0.1

Type RM Length L Ch R = 1 ,18479   ,509,509,509
BEGIN DESCRIPTION:
YEAGER CREEK 33.0
END DESCRIPTION:
XS GIS Cut Line= 4
      2942812.13     10044925.43      2943232.26     10045467.09
      2944343.37     10045644.17       2945141.2     10045939.02
#Sta/Elev= 30
  3771.2 1219.64  3888.4 1214.31  3952.7 1206.56  4025.5 1203.01  4148.3 1194.82
  4245.1 1189.04  4301.2    1169  4344.7 1158.96  4359.2 1157.88  4373.6 1153.34
  4394.5  1142.8  4429.8 1136.32  4534.8 1132.19  4807.3 1129.76  4837.7 1124.73
  4845.5 1121.99  4894.1 1118.58    4980 1117.99  5006.8  1112.8  5009.5  1112.3
  5012.8  1112.8    5037 1121.42  5060.4 1124.92  5090.8 1136.05  5111.1 1150.61
  5248.5 1154.58  5955.5 1164.58    6099 1166.72  6411.8 1178.33  6432.4  1178.9
#Mann= 9 ,-1 , 0
  3771.2     .16       0  4025.5      .1       0  4148.3     .16       0
  4894.1      .1       0  5006.8     .07       0  5012.8      .1       0
  5248.5     .05       0  5955.5      .1       0  6411.8     .05       0
Bank Sta=4837.7,5060.4
XS Rating Curve= 0 ,0
Exp/Cntr=0.3,0.1

Type RM Length L Ch R = 1 ,17970   ,190,190,190
BEGIN DESCRIPTION:
YEAGER CREEK 32.0
END DESCRIPTION:
XS GIS Cut Line= 4
      2942263.52     10045696.25      2943336.43      10045953.2
      2943937.12     10046119.86      2945054.28     10046043.54
#Sta/Elev= 30
  3580.6 1199.12  3647.4 1198.08  3811.9 1187.89  3848.4 1182.84    4153 1162.24
  4212.9  1158.5  4243.8 1148.96  4284.9 1144.33  4336.3 1141.65  4346.6 1143.29
  4387.7 1138.85  4480.3 1137.62  4682.3 1126.37  4872.8 1120.59  4955.8 1117.69
  5005.3 1111.75  5008.1 1111.25  5011.3 1111.75  5028.4 1119.71  5042.6 1126.91
  5059.7 1127.83  5132.2  1129.6  5160.8 1132.98  5215.2 1146.56    5262 1150.99
  5579.6 1160.01  5779.5 1164.64  6056.4 1170.13  6353.9 1176.95    6427  1179.1
#Mann= 11 ,-1 , 0
  3580.6      .1       0    4153     .16       0  5005.3     .07       0
  5011.3     .16       0  5059.7     .05       0  5160.8     .16       0
    5262     .05       0  5579.6      .1       0  5779.5     .05       0
  6056.4      .1       0  6353.9     .05       0
Bank Sta=4872.8,5028.4
XS Rating Curve= 0 ,0
Exp/Cntr=0.3,0.1

Type RM Length L Ch R = 1 ,17780   ,195,195,195
BEGIN DESCRIPTION:
YEAGER CREEK 31.0
END DESCRIPTION:
XS GIS Cut Line= 2
      2942457.93     10045974.03      2944394.43      10046352.3
#Sta/Elev= 30
  3920.2 1178.97  4379.7 1159.17  4440.4 1156.15  4501.5 1137.94  4517.7 1135.24
  4883.6 1119.39  4970.2 1115.41  4988.8 1110.36  4991.6 1109.86  4994.8 1110.36
  5031.3 1114.48  5051.7 1121.08  5077.6 1126.33  5177.3 1127.55    5296 1128.84
  5326.8 1131.25  5352.7 1137.02  5357.8 1135.68  5376.7 1140.47  5404.2 1147.33
  5409.3 1145.89  5455.8 1151.32  5507.3 1152.09  5512.4 1149.42  5652.9 1157.06
  5683.4 1153.43  5713.6 1158.15  5775.5 1160.08  5875.2 1160.89  5893.3 1160.91
#Mann= 9 ,-1 , 0
  3920.2      .1       0  4379.7     .08       0  4988.8     .07       0
  4994.8     .08       0  5077.6     .05       0  5177.3     .08       0
  5376.7      .1       0  5775.5     .08       0  5875.2      .1       0
Bank Sta=4883.6,5051.7
XS Rating Curve= 0 ,0
Exp/Cntr=0.3,0.1

Type RM Length L Ch R = 1 ,17585   ,514,514,514
BEGIN DESCRIPTION:
YEAGER CREEK 30.0
END DESCRIPTION:
XS GIS Cut Line= 3
      2942385.03     10046147.64      2944211.43     10046487.92
      2944363.86     10046491.38
#Sta/Elev= 30
  3963.5 1168.76  4587.5 1157.14  4607.8 1155.28  4623.9 1150.42  4628.9 1151.51
  4676.6  1135.1  4681.7 1135.64  4689.2 1132.26  4709.6 1128.21  4760.4 1127.16
    4852 1119.67    4913 1117.59  4950.4 1115.63  4984.2 1109.76  5000.1 1109.15
  5002.9 1108.65  5006.1 1109.15  5024.9 1114.89  5055.4 1117.43  5126.6 1123.55
    5277 1129.08  5334.8 1126.51  5523.3 1128.63  5574.2 1132.77  5603.5 1137.53
  5608.6 1136.56  5645.4 1146.93  5661.3 1149.74  5766.8 1154.72  5973.8 1156.52
#Mann= 3 ,-1 , 0
  3963.5     .05       0  5000.1     .04       0  5006.1     .05       0
Bank Sta=4913,5055.4
XS Rating Curve= 0 ,0
Exp/Cntr=0.3,0.1

Type RM Length L Ch R = 1 ,17071   ,807,807,807
BEGIN DESCRIPTION:
YEAGER CREEK 29.0
END DESCRIPTION:
XS GIS Cut Line= 4
      2941680.14     10046533.05      2942690.59     10046845.56
      2943763.51     10046786.53       2944363.8     10046515.88
#Sta/Elev= 30
  3359.5 1184.66  3526.9 1177.57  3956.8 1170.81  4016.9 1168.17    4060 1168.69
    4120 1164.68  4499.4 1159.95    4591 1158.99  4735.5 1156.87  4875.7 1149.36
  4908.2 1140.61  4925.8 1130.47  4945.8 1115.63  4952.6 1113.68  4992.9 1107.77
  4995.7 1107.27  4998.9 1107.77    5056 1111.34  5136.1 1112.85  5156.2 1115.62
  5216.3 1125.64  5296.2 1126.81  5395.2 1124.26  5494.5 1126.21  5829.3 1131.11
  5869.8  1133.6  5904.2 1145.31  5927.4 1150.46  5983.2 1152.78  6150.2 1156.38
#Mann= 13 ,-1 , 0
  3359.5      .1       0  3526.9     .05       0  3956.8      .1       0
  4499.4     .05       0    4591      .1       0  4952.6     .05       0
  4992.9    .033       0  4998.9     .05       0  5296.2      .1       0
  5395.2     .05       0  5494.5      .1       0  5869.8     .16       0
  5983.2     .05       0
Bank Sta=4945.8,5156.2
XS Rating Curve= 0 ,0
Exp/Cntr=0.3,0.1

Type RM Length L Ch R = 1 ,16264   ,60,60,60
BEGIN DESCRIPTION:
Mapping XS 194e1812
END DESCRIPTION:
XS GIS Cut Line= 4
      2941666.83     10046580.93      2942951.52     10047496.71
       2943628.6     10047600.87      2944334.78     10048060.11
#Sta/Elev= 30
  3202.8 1187.06  3381.2 1184.83  3604.3 1183.11  4166.3 1165.93  4421.7 1161.78
  4489.6    1154  4518.8 1146.62    4568 1126.86  4593.4 1121.22  4626.1 1117.96
    4828 1115.33  4861.5 1115.96  4878.6  1122.5  4898.8 1116.35  4949.4 1107.82
  5027.3 1106.09  5030.1 1105.59  5033.3 1106.09  5151.7 1108.73  5212.5 1116.52
  5371.2 1122.02  5470.3  1125.1  5490.2 1126.48    5699 1139.61  5727.8 1138.76
  5842.7 1152.01  5914.4 1161.97  6002.2 1184.29  6103.6 1204.28  6307.9 1208.45
#Mann= 12 ,-1 , 0
  3202.8      .1       0  3381.2     .05       0  3604.3      .1       0
  4421.7     .16       0  4593.4     .05       0  5027.3    .033       0
  5033.3     .05       0  5371.2      .1       0  5470.3     .16       0
  5490.2      .1       0  5842.7     .05       0  5914.4      .1       0
#XS Ineff= 2 , 0
         4877.27 1122.68
Permanent Ineff=
       T       T
Bank Sta=4898.8,5212.5
XS Rating Curve= 0 ,0
Exp/Cntr=0.3,0.1

Type RM Length L Ch R = 1 ,16204   ,59,59,59
BEGIN DESCRIPTION:
YEAGER CREEK 28.0
END DESCRIPTION:
XS GIS Cut Line= 4
      2941638.49     10046647.63      2942944.07     10047553.89
      2943582.96     10047658.06      2944304.33     10048157.47
#Sta/Elev= 30
    3195 1190.45  3371.5 1187.13  3384.5  1187.1  3501.1 1186.15  3534.2 1185.16
  4434.3  1157.8  4478.2 1148.21  4534.9 1126.37  4558.6 1121.05  4737.5 1115.24
  4859.7 1115.11  4875.7 1119.81  4890.1  1120.2  4930.6 1117.02  5040.5 1115.02
  5057.1 1114.46  5059.8 1113.96  5063.1 1114.46  5095.1 1115.24 5106.03 1116.99
    5113 1119.54  5339.7 1120.71  5631.2 1134.34  5784.6 1144.06  5855.5 1152.97
  5912.9 1162.42  5972.4  1180.9    6065 1203.62  6157.5 1210.26    6309 1211.64
#Mann= 14 ,-1 , 0
    3195      .1       0  3371.5     .05       0  3384.5      .1       0
  3501.1     .05       0  3534.2      .1       0  4434.3     .16       0
  4558.6     .05       0  5040.5      .1       0  5057.1    .033       0
  5063.1      .1       0  5095.1     .05       0  5339.7      .1       0
  5631.2     .05       0  5855.5      .1       0
#XS Ineff= 2 , 0
         4899.65 1120.22
Permanent Ineff=
       T       T
Bank Sta=4930.6,5106.03
XS Rating Curve= 0 ,0
Exp/Cntr=0.3,0.1

Type RM Length L Ch R = 1 ,16145   ,385,385,385
BEGIN DESCRIPTION:
YEAGER CREEK 27.0
END DESCRIPTION:
XS GIS Cut Line= 4
      2941627.78     10046732.85       2942895.1     10047609.56
      2943572.18     10047709.38      2944123.12     10048399.14
#Sta/Elev= 30
  3205.5 1193.07    3222 1192.88  3403.1  1190.1  3406.2 1190.03  3571.7 1184.12
  4371.8 1156.57  4407.6 1153.71    4452 1140.76  4484.9 1128.13    4515 1120.56
  4543.9  1119.1  4770.1 1114.34  4911.6 1115.52  4931.9 1111.47  4966.5 1104.92
  4999.6 1101.19  5002.4 1100.69  5005.6 1101.19    5081 1103.11  5103.7 1109.89
  5200.4 1115.63  5339.8 1120.85  5571.5 1131.84  5737.1 1137.19  5830.2 1142.51
  5961.5  1166.7  6078.4 1201.99  6116.3 1208.84  6212.7 1215.54  6313.7 1217.63
#Mann= 17 ,-1 , 0
  3205.5      .1       0    3222     .05       0  3403.1      .1       0
  3406.2     .05       0  3571.7      .1       0    4452     .16       0
  4484.9     .05       0  4966.5      .1       0  4999.6     .07       0
  5005.6      .1       0  5200.4     .05       0  5339.8      .1       0
  5571.5     .05       0  5737.1      .1       0  5961.5     .16       0
  6116.3      .1       0  6212.7     .16       0
#XS Ineff= 2 ,-1
  3205.5  4907.1 1116.07 5220.39 5255.73 1116.95
Permanent Ineff=
       T       T
Bank Sta=4931.9,5103.7
XS Rating Curve= 0 ,0
Exp/Cntr=0.3,0.1

Type RM Length L Ch R = 1 ,15760   ,952,952,952
BEGIN DESCRIPTION:
YEAGER CREEK 26.0
END DESCRIPTION:
XS GIS Cut Line= 4
      2941499.66     10046984.47      2942881.57     10047901.11
      2943395.46     10048248.34      2944207.96     10048692.78
#Sta/Elev= 30
  3153.9 1197.91  3156.6 1197.89  3255.9 1192.97  3325.4 1190.04  3354.7 1182.23
  3389.9 1181.08  3486.2 1183.41  4061.9 1163.64    4177 1151.77  4203.9 1146.02
  4278.9 1138.57    4336 1126.12  4414.2 1120.52  4765.2 1111.31  4898.1 1108.67
    5003 1101.12  5005.7 1100.62    5009 1101.12    5042 1101.96 5054.26 1108.71
  5113.9 1113.63  5289.9 1115.43  5292.5 1115.18  5446.2 1118.14  5531.2 1123.35
  5815.1 1169.96  5929.5 1195.11  5992.2 1207.91    6144 1217.37  6358.5 1218.19
#Mann= 19 ,-1 , 0
  3153.9     .05       0  3156.6      .1       0  3255.9     .05       0
  3354.7      .1       0  3389.9     .05       0  3486.2      .1       0
  4061.9     .16       0    4177     .05       0  4203.9      .1       0
  4765.2     .05       0    5003    .035       0    5009     .05       0
  5289.9      .1       0  5292.5     .05       0  5446.2      .1       0
  5531.2     .16       0  5815.1      .1       0  5929.5     .16       0
    6144      .1       0
#XS Ineff= 2 ,-1
 5071.81 5099.34  1111.1 5122.93  6358.5 1113.71
Permanent Ineff=
       T       T
Bank Sta=4898.1,5054.26
XS Rating Curve= 0 ,0
Exp/Cntr=0.3,0.1

Type RM Length L Ch R = 1 ,14808   ,1041,1041,1041
BEGIN DESCRIPTION:
YEAGER CREEK 24.0
END DESCRIPTION:
XS GIS Cut Line= 4
      2941027.39     10048192.78       2942402.4     10048734.45
      2944048.23     10048831.67      2944374.59     10048949.71
#Sta/Elev= 30
    2962 1211.64  3441.7 1181.23  3667.2 1171.37  3988.7 1157.01  4151.1 1145.64
    4370 1135.91    4584 1124.72  4886.7 1111.13  4918.6 1106.15  4936.8 1101.34
    5064 1101.21  5066.8 1100.71    5070 1101.21  5097.1 1101.33 5113.64 1106.13
  5127.1 1108.51  5567.9 1111.11  5694.7 1118.15  5718.1  1121.1  5748.2 1129.52
  5798.3 1154.36  5838.4 1169.68  5866.3 1186.31  5871.3 1184.97  5888.4 1195.76
  5928.5  1207.4  5970.1 1212.94  6008.6 1217.01    6107 1220.39  6435.6 1225.03
#Mann= 9 ,-1 , 0
    2962     .05       0  3667.2      .1       0    4370     .05       0
    4584      .1       0  4918.6     .05       0    5064    .033       0
    5070     .05       0  5694.7     .16       0  5970.1      .1       0
#XS Ineff= 2 , 0
                         5256.29         1108.86
Permanent Ineff=
       T       T
Bank Sta=4918.6,5113.64
XS Rating Curve= 0 ,0
Exp/Cntr=0.3,0.1

Type RM Length L Ch R = 1 ,13767   ,790,790,790
BEGIN DESCRIPTION:
YEAGER CREEK 22.0
END DESCRIPTION:
XS GIS Cut Line= 4
      2941082.93     10048505.27      2942798.23     10049678.89
      2943944.07     10049748.34      2944228.78     10049685.84
#Sta/Elev= 30
  2490.8 1196.16    2939 1173.16    2990 1171.09    3588 1146.46  3723.1 1137.61
  3775.5 1125.82  3809.8 1118.01  3824.7 1119.66  3897.4 1108.03  4198.5 1103.54
  4723.1 1103.76  4821.7 1104.02    4880 1103.81  4896.1 1096.48  5007.2 1093.65
    5010 1093.15  5013.2 1093.65  5040.3 1097.01  5046.3 1097.32  5140.5 1104.63
  5220.6 1117.64  5320.8 1150.26  5380.9 1163.71    5451 1189.21  5511.8 1202.34
  5562.3 1211.62  5702.6 1221.26  5935.8 1234.84    5994 1241.04  6008.6 1245.56
#Mann= 13 ,-1 , 0
  2490.8     .05       0    2939      .1       0    2990     .05       0
  3775.5      .1       0  3897.4     .05       0  4723.1     .16       0
  4821.7     .05       0  5007.2    .033       0  5013.2     .05       0
  5046.3     .16       0  5511.8     .05       0  5702.6      .1       0
  5935.8     .05       0
#XS Ineff= 2 , 0
         4860.31 1104.91
Permanent Ineff=
       T       T
Bank Sta=4896.1,5040.3
XS Rating Curve= 0 ,0
Exp/Cntr=0.3,0.1

Type RM Length L Ch R = 1 ,12977   ,799,799,799
BEGIN DESCRIPTION:
YEAGER CREEK 21.0
END DESCRIPTION:
XS GIS Cut Line= 3
      2941062.14     10050574.72      2942687.12     10050387.23
      2944304.34     10049894.43
#Sta/Elev= 30
  3097.3 1169.37  3588.8 1139.81  3677.8 1120.68  3717.7 1104.05  3768.1 1097.44
  4272.2 1100.45  4485.9 1105.16  4571.6 1104.52  4613.6  1099.8  4714.3 1104.82
    4773 1094.74  4877.5 1090.97  4891.3 1087.68  5069.6 1082.17  5072.3 1081.67
  5075.6 1082.17  5094.1 1084.56  5143.5 1087.86  5236.3 1105.08  5307.7 1134.94
  5378.6 1154.57  5437.4 1159.92  5487.5 1165.59  5591.7 1188.56  5758.5  1211.1
  5943.7 1217.89  6015.7 1218.95  6071.8 1219.12  6340.5 1226.23  6423.7 1231.13
#Mann= 15 ,-1 , 0
  3097.3     .05       0  4272.2     .16       0  4485.9     .05       0
  4571.6      .1       0    4773     .16       0  4877.5     .05       0
  5069.6    .033       0  5075.6     .05       0  5094.1      .1       0
  5437.4     .05       0  5758.5      .1       0  5943.7     .05       0
  6015.7      .1       0  6071.8     .05       0  6340.5      .1       0
Bank Sta=4891.3,5143.5
XS Rating Curve= 0 ,0
Exp/Cntr=0.3,0.1

Type RM Length L Ch R = 1 ,12178   ,1044,1044,1044
BEGIN DESCRIPTION:
YEAGER CREEK 19.0
END DESCRIPTION:
XS GIS Cut Line= 2
       2941214.9     10051060.84      2944131.59     10051067.78
#Sta/Elev= 30
  3104.7 1150.86  3214.7 1147.57  3459.2 1138.64  3572.9 1132.55  3788.3 1119.52
  3828.3 1114.96  3912.9 1098.08  4018.3 1091.53  4168.3 1094.59  4248.3  1084.5
  4858.3 1087.12  4881.8  1082.3  4935.3 1082.02    4938 1081.52  4941.3 1082.02
  5088.3 1083.28  5108.3 1087.32  5128.3 1094.25  5177.7 1096.86  5228.3 1098.07
  5276.4  1121.2  5338.3 1152.94  5417.6 1161.71    5431 1164.25  5578.3 1185.65
  5652.6  1192.4  5669.7 1193.47  5728.3 1197.58  5808.3 1211.47  6021.4 1216.57
#Mann= 14 ,-1 , 0
  3104.7      .1       0  3214.7     .05       0  3459.2      .1       0
  3572.9     .05       0  3912.9      .1       0  4881.8     .05       0
  4935.3    .033       0  4941.3     .05       0  5177.7     .16       0
  5276.4      .1       0  5417.6     .05       0    5431      .1       0
  5652.6     .05       0  5669.7      .1       0
#XS Ineff= 2 ,-1
 3979.79 4138.59 1093.51 4213.03 4849.07 1087.64
Permanent Ineff=
       T       T
Bank Sta=4858.3,5108.3
XS Rating Curve= 0 ,0
Exp/Cntr=0.3,0.1

Type RM Length L Ch R = 1 ,11134   ,213,213,213
BEGIN DESCRIPTION:
YEAGER CREEK 17.0
END DESCRIPTION:
XS GIS Cut Line= 3
      2941159.34     10052012.23      2943249.62     10051991.39
      2944291.31      10051401.1
#Sta/Elev= 30
  3347.2 1143.31  3462.3 1139.77  3569.3 1137.25  3686.3 1129.48  3758.4  1129.2
  3927.8  1127.4  4106.4 1121.47  4236.4 1102.18  4295.9 1098.79  4296.6 1098.76
  4426.4 1094.44  4466.4 1099.57  4506.4 1099.58  4548.1 1091.91 4759.14 1085.81
  4786.4 1082.83  5163.4 1082.61  5166.2 1082.11  5169.4 1082.61 5192.53 1085.85
  5239.1 1099.67  5337.8 1129.69  5466.4 1153.73  5629.5  1167.8  5728.2 1178.33
  5765.7 1186.52  5889.7 1194.69  6013.8 1209.86  6315.4 1218.21  6634.9 1215.02
#Mann= 14 ,-1 , 0
  3347.2     .16       0  3462.3     .05       0  3569.3      .1       0
  3758.4     .05       0  3927.8      .1       0  4295.9     .05       0
  4296.6      .1       0  4548.1     .05       0  5163.4    .033       0
  5169.4     .05       0  5239.1     .16       0  5337.8      .1       0
  5466.4     .05       0  5629.5      .1       0
#XS Ineff= 2 , 0
          4745.6 1087.57
Permanent Ineff=
       T       T
Bank Sta=4759.14,5192.53
XS Rating Curve= 0 ,0
Exp/Cntr=0.3,0.1

Type RM Length L Ch R = 1 ,10921   ,87,87,87
BEGIN DESCRIPTION:
Mapping XS 10b27ea1
END DESCRIPTION:
XS GIS Cut Line= 5
      2941193.89     10052182.09      2942535.07     10052158.65
       2943055.9     10052257.61      2943423.09     10052143.02
       2944292.9     10051455.51
#Sta/Elev= 30
    3392 1147.08  3593.7 1133.99  3846.6 1125.69  3896.7 1115.62  3926.7 1123.24
  3987.2 1123.23  3991.3 1123.07  4086.7 1121.32  4152.1 1113.42  4349.1 1092.77
  4436.7 1092.29  4496.7 1100.46  4551.6  1095.1  4586.8 1085.68  4643.8 1080.79
  4646.5 1080.29  4649.8 1080.79  4749.3 1083.82  4949.7 1082.61  5024.7 1082.68
  5247.4 1082.18  5287.2 1083.86  5560.8 1151.56  5669.2 1160.91  5760.5 1168.41
  5762.1 1168.43  5914.7 1186.39  6087.1 1194.65    6285 1212.77  6756.9 1214.47
#Mann= 18 ,-1 , 0
    3392     .05       0  3593.7      .1       0  3987.2     .05       0
  3991.3      .1       0  4152.1     .05       0  4349.1      .1       0
  4551.6     .05       0  4643.8    .033       0  4649.8     .05       0
  4749.3      .1       0  4949.7     .05       0  5024.7      .1       0
  5247.4     .16       0  5560.8      .1       0  5669.2     .05       0
  5760.5      .1       0  5762.1     .05       0  6087.1      .1       0
#XS Ineff= 2 , 0
         4716.45 1085.74
Permanent Ineff=
       T       T
Bank Sta=4749.3,5287.2
XS Rating Curve= 0 ,0
Exp/Cntr=0.3,0.1

Type RM Length L Ch R = 1 ,10834   ,96,96,96
BEGIN DESCRIPTION:
Mapping XS 91e1d71d
END DESCRIPTION:
XS GIS Cut Line= 5
      2941230.35     10052221.15       2942493.4     10052208.13
      2942897.05     10052320.11      2943355.38     10052291.46
      2944269.45     10051512.81
#Sta/Elev= 30
  3414.5 1146.36  3586.7  1134.7  3832.6 1126.15  3902.6 1111.98  4050.3 1112.69
  4152.7 1110.58  4262.7 1096.41  4359.9 1094.42  4422.7 1092.04  4482.7 1100.99
  4535.5 1096.51  4582.7 1084.56  4734.3 1081.05  4890.4 1075.57  5001.6 1069.89
  5004.3 1069.39  5007.6 1069.89  5024.1 1070.67  5077.2 1076.59    5238 1081.55
  5253.2 1082.15  5388.5  1095.3  5653.7 1155.09  5661.7 1155.57  5842.4 1168.47
  5904.3 1174.94  6215.7 1198.75  6370.3 1212.42  6393.5 1212.94  6756.5 1214.63
#Mann= 18 ,-1 , 0
  3414.5     .05       0  3586.7      .1       0  4050.3     .05       0
  4359.9      .1       0  4535.5     .05       0  4734.3      .1       0
  5001.6     .07       0  5007.6      .1       0  5024.1     .05       0
    5238      .1       0  5253.2     .16       0  5653.7      .1       0
  5661.7     .05       0  5842.4      .1       0  5904.3     .05       0
  6215.7      .1       0  6370.3     .05       0  6393.5      .1       0
#XS Ineff= 3 ,-1
 4608.34 4712.59 1082.22 4714.91  4725.4 1081.25 4749.28 4765.58 1079.77
Permanent Ineff=
       T       T       T
Bank Sta=4890.4,5077.2
XS Rating Curve= 0 ,0
Exp/Cntr=0.3,0.1

Type RM Length L Ch R = 1 ,10738   ,735,735,735
BEGIN DESCRIPTION:
Mapping XS 4701b3b0
END DESCRIPTION:
XS GIS Cut Line= 5
      2941235.58     10052320.97      2942628.82     10052329.66
      2942910.94      10052399.1      2943362.32     10052360.04
      2944303.78     10051631.17
#Sta/Elev= 30
  3420.2 1148.83  3633.7 1132.58  3991.9 1122.28  4053.1 1114.23  4193.1  1110.8
  4423.1  1092.2  4473.1 1101.64  4530.9 1099.71  4573.1 1087.62  4642.7 1081.91
  4763.1 1071.79  4850.3 1076.17  4882.2  1069.6  4884.9  1069.1  4888.2  1069.6
  5008.8 1069.72  5080.9 1075.64  5257.5 1081.72  5299.8 1081.75  5421.8 1088.58
  5573.4  1121.1  5594.2 1130.75  5690.2 1154.33  5785.7 1161.41  5913.3 1167.72
  6052.3 1175.17  6298.6 1197.33  6417.3 1206.02  6438.8 1207.76  6747.7 1209.85
#Mann= 17 ,-1 , 0
  3420.2     .05       0  3633.7      .1       0  3991.9     .05       0
  4530.9      .1       0  4642.7     .05       0  4882.2    .033       0
  4888.2     .05       0  5257.5      .1       0  5299.8     .05       0
  5421.8     .16       0  5690.2      .1       0  5785.7     .05       0
  5913.3      .1       0  6052.3     .05       0  6298.6      .1       0
  6417.3     .05       0  6438.8      .1       0
#XS Ineff= 1 ,-1
 5220.73 5251.41 1081.17
Permanent Ineff=
       T
Bank Sta=4850.3,5080.9
XS Rating Curve= 0 ,0
Exp/Cntr=0.3,0.1

Type RM Length L Ch R = 1 ,10003   ,592,592,592
BEGIN DESCRIPTION:
YEAGER CREEK 16.0
END DESCRIPTION:
XS GIS Cut Line= 4
      2941687.01     10053158.65      2943132.29     10053050.14
      2943501.21     10052286.25      2943769.28     10052208.43
#Sta/Elev= 30
  3369.8 1133.47  3401.9 1131.51  3549.3 1125.75  3600.4 1124.28  3622.6 1123.69
  3839.3 1118.21  3962.9 1114.41    3993 1107.71  4143.4 1109.92  4369.6 1102.02
  4414.2  1096.6  4544.6 1088.59  4819.1 1081.07    4872 1075.35  4881.8 1070.89
  4894.6 1069.79  4945.4 1069.65  4948.2 1069.15  4951.4 1069.65  5024.7 1070.75
  5052.9 1074.89    5307 1080.07  5397.4 1087.15  5447.5 1099.01  5561.2 1134.12
  5578.3 1135.73  5606.4 1145.75  5638.8 1152.91  5770.1  1161.1  5946.6 1162.85
#Mann= 11 ,-1 , 0
  3369.8     .05       0  3401.9     .16       0  3549.3     .05       0
  3600.4      .1       0  3622.6     .05       0  3839.3      .1       0
  4369.6     .05       0  4945.4    .033       0  4951.4     .05       0
  5447.5     .16       0  5638.8      .1       0
Bank Sta=4872,5052.9
XS Rating Curve= 0 ,0
Exp/Cntr=0.3,0.1

Type RM Length L Ch R = 1 ,9411    ,73,73,73
BEGIN DESCRIPTION:
Mapping XS 17eda15b
END DESCRIPTION:
XS GIS Cut Line= 4
      2941705.16     10053201.62      2943744.18     10053175.58
      2943785.85     10052956.83      2943744.18     10052370.87
#Sta/Elev= 30
  2819.6 1132.39  2831.5 1131.86  3002.5 1124.96  3284.2 1117.54  3402.9    1114
    3423 1108.66    3493 1108.21    3513 1111.71  3820.8 1101.65    3863 1096.98
    4203 1081.91    4333 1083.04    4563 1073.39  4693.1 1080.79  4783.1 1074.68
  4907.4 1073.38  4931.9 1069.96  5114.4 1069.61  5117.1 1069.11  5120.4 1069.61
    5253 1069.82  5263.8  1073.1  5304.7 1078.15  5355.2 1081.45  5393.7 1097.59
  5398.7 1096.75  5465.5 1126.55  5544.6 1145.06  5565.8 1148.98  5668.9 1153.36
#Mann= 9 ,-1 , 0
  2819.6     .05       0  2831.5     .16       0  3002.5     .05       0
  3284.2      .1       0  3820.8     .05       0  5114.4    .035       0
  5120.4     .05       0  5304.7     .16       0  5544.6      .1       0
#XS Ineff= 2 ,-1
  4387.3 4683.49 1080.75 4759.61 4901.29 1074.77
Permanent Ineff=
       T       T
Bank Sta=4907.4,5263.8
XS Rating Curve= 0 ,0
Exp/Cntr=0.3,0.1

Type RM Length L Ch R = 1 ,9338    ,167,167,167
BEGIN DESCRIPTION:
Mapping XS b85bf989
END DESCRIPTION:
XS GIS Cut Line= 4
      2941697.27     10053225.05      2943793.66     10053204.22
      2943871.79     10052925.58      2943905.38     10052320.59
#Sta/Elev= 30
  2736.7 1132.92  2755.5 1132.06  2914.2 1125.37  3214.1 1117.27  3317.9 1115.09
  3357.9 1108.44  3567.9 1109.17  3751.4  1098.7    4058 1085.88    4108 1079.96
    4318 1080.98    4488 1072.21    4598 1080.14    4718 1074.09  4885.6 1073.66
  4934.6 1066.02  4937.3 1065.52  4940.6 1066.02  4943.2 1070.97  4958.3 1066.77
  4977.3 1070.84  4989.5 1066.17  5095.1 1071.49  5254.6 1070.31  5309.5 1077.83
    5495 1100.66    5525 1117.64  5574.9 1134.09  5625.2 1145.43  5728.5 1155.19
#Mann= 9 ,-1 , 0
  2736.7     .05       0  2755.5     .16       0  2914.2     .05       0
  3214.1      .1       0  3751.4     .05       0  4934.6    .035       0
  4940.6     .05       0  5309.5     .16       0  5574.9      .1       0
Bank Sta=4934.6,4940.6
XS Rating Curve= 0 ,0
Exp/Cntr=0.3,0.1

Type RM Length L Ch R = 1 ,9171    ,267,267,267
BEGIN DESCRIPTION:
Mapping XS d8c4d111
END DESCRIPTION:
XS GIS Cut Line= 4
      2941710.32     10053243.28      2943827.52     10053219.85
      2944393.22     10052888.12      2944964.77     10052703.66
#Sta/Elev= 30
  2703.6 1132.99  2708.6 1132.46  2857.9 1125.68  3171.6 1117.17  3271.8 1115.19
  3311.8 1108.54  3391.8 1111.83  3521.8 1108.84  3708.9 1097.29  3781.8 1095.23
  3881.8 1083.57  3941.8 1085.54  4141.8 1078.03  4271.8 1080.59  4431.9 1071.97
  4541.9 1078.38  4841.2 1073.08  4969.7 1064.55  4972.5 1064.05  4975.7 1064.55
  5097.2 1065.51  5294.6 1077.58  5360.7 1089.73  5433.3 1123.35  5477.9  1130.9
  5789.2 1155.14  5843.7 1158.37  5934.9 1164.11  6025.8 1178.27  6077.3 1181.59
#Mann= 11 ,-1 , 0
  2703.6     .05       0  2708.6     .16       0  2857.9     .05       0
  3171.6      .1       0  3708.9     .05       0  4969.7    .035       0
  4975.7     .05       0  5360.7     .16       0  5477.9     .05       0
  5789.2      .1       0  5843.7     .05       0
Bank Sta=4969.7,4975.7
XS Rating Curve= 0 ,0
Exp/Cntr=0.3,0.1

Type RM Length L Ch R = 1 ,8904    ,705,705,705
BEGIN DESCRIPTION:
YEAGER CREEK 15.0
END DESCRIPTION:
XS GIS Cut Line= 3
      2941700.97     10053255.28      2943784.34     10053269.17
      2944873.07     10053518.81
#Sta/Elev= 30
  2591.4 1133.26  2605.2 1132.53  2746.9 1125.73  3070.9 1116.87  3168.9 1115.61
  3208.9 1108.88  3288.9 1111.51  3408.9 1108.61  3612.3  1096.4  3668.9 1093.57
  3748.9 1081.51  3928.9 1075.75  4158.9 1077.13  4318.9 1070.26  4448.9 1074.96
  4750.9 1071.78  5045.4 1064.94  5048.1 1064.44  5051.4 1064.94  5077.6 1065.51
    5110 1066.61  5117.7 1068.38 5118.38 1071.89  5130.5 1086.26  5177.9 1116.82
  5213.7 1132.85  5278.1 1140.79  5390.4 1149.71  5619.8 1156.66  5791.8  1167.7
#Mann= 11 ,-1 , 0
  2591.4     .05       0  2605.2     .16       0  2746.9     .05       0
  3070.9      .1       0  3612.3     .05       0  5045.4    .033       0
  5051.4     .05       0  5077.6      .1       0  5177.9     .05       0
  5278.1      .1       0  5619.8     .05       0
#XS Ineff= 2 ,-1
 3872.25 4087.47 1076.79  4195.9  4448.9 1074.88
Permanent Ineff=
       T       T
Bank Sta=4750.9,5118.38
XS Rating Curve= 0 ,0
Exp/Cntr=0.3,0.1

Type RM Length L Ch R = 1 ,8571    ,291,291,291
BEGIN DESCRIPTION:
Mapping XS ad354517
END DESCRIPTION:
XS GIS Cut Line= 4
      2941746.51     10053341.46      2943365.91     10053340.03
      2944212.55     10053564.66      2944689.18     10053549.79
#Sta/Elev= 30
  2933.4 1130.72  3019.5 1126.77    3345 1116.83  3465.4 1115.08  3505.4 1109.39
  3695.4 1108.43  3925.5 1091.02  4025.4  1075.3  4515.8 1068.15  4766.3 1068.89
  4895.2  1069.3  4945.6 1064.61  4948.3 1064.11  4951.6 1064.61  5083.1  1069.4
  5155.5 1064.98  5181.5 1071.26  5196.9 1067.08  5206.4 1072.37  5217.6 1086.66
  5238.3 1088.92    5259 1106.17  5313.4 1113.08  5367.1 1117.31  5414.2 1131.18
  5483.2 1134.34    5613 1145.72  5627.2 1145.18  5882.8 1157.38  5905.6 1158.29
#Mann= 14 ,-1 , 0
  2933.4     .16       0  3019.5     .05       0    3345      .1       0
  3925.5     .05       0  4515.8     .16       0  4766.3     .05       0
  4945.6    .033       0  4951.6     .05       0  5181.5      .1       0
  5313.4     .05       0  5483.2      .1       0    5613     .05       0
  5627.2      .1       0  5882.8     .05       0
Bank Sta=4945.6,4951.6
XS Rating Curve= 0 ,0
Exp/Cntr=0.3,0.1

Type RM Length L Ch R = 1 ,8280    ,186,186,186
BEGIN DESCRIPTION:
Mapping XS 8d80a9d9
END DESCRIPTION:
XS GIS Cut Line= 4
      2941733.81      10053313.6      2943353.56     10053383.91
      2943615.68     10053628.63      2944543.59     10053592.24
#Sta/Elev= 30
  3150.3 1131.53  3253.9  1126.5  3577.4 1116.76  3705.5 1114.45  3735.5 1109.39
  3815.6 1111.46  3960.6 1107.11  4159.6 1090.91  4175.9 1089.53    4216 1077.67
    4256  1073.2  4635.6    1067  4815.1 1068.43  4913.2 1064.58    4916 1064.08
  4919.2 1064.58  5020.5 1064.73  5072.1 1065.32  5086.2 1067.83  5093.1 1075.04
  5100.4 1070.05  5107.2 1083.79  5114.6 1085.98  5353.1 1092.36  5483.5 1103.87
  5663.4 1116.43  5723.4 1130.36  5780.2 1133.77  5913.6 1145.59  6058.8 1153.69
#Mann= 11 ,-1 , 0
  3150.3     .16       0  3253.9     .05       0  3577.4      .1       0
  4159.6     .05       0  4635.6     .16       0  4815.1     .05       0
  4913.2    .033       0  4919.2     .05       0  5020.5      .1       0
  5483.5     .05       0  5780.2      .1       0
Bank Sta=4913.2,4919.2
XS Rating Curve= 0 ,0
Exp/Cntr=0.3,0.1

Type RM Length L Ch R = 1 ,8094    ,167,167,167
BEGIN DESCRIPTION:
Mapping XS 8d4a81cf
END DESCRIPTION:
XS GIS Cut Line= 5
        2941692.     10053396.66      2943087.03     10053428.24
      2943245.73     10053473.48      2943406.76     10053668.57
      2944444.29     10053654.38
#Sta/Elev= 30
  3289.3 1138.48  3325.8 1131.92  3418.3 1127.14  3739.6 1117.14  3915.9 1109.96
    4086 1108.56  4353.2  1090.4  4436.1 1068.65  4721.5  1065.8  4873.5 1062.75
  4909.9 1065.43  4929.5 1061.87  4937.4 1056.58  4943.8 1060.13  4948.7 1056.22
  4951.4 1055.72  4954.7 1056.22  4958.2 1061.36    4966 1058.59  4972.5 1063.14
  4986.9 1057.39  4993.3 1064.16  5050.7 1065.09  5085.9 1078.21  5184.4 1078.54
  5224.4 1083.31  5544.4 1093.03  5864.4 1115.69  5954.5 1132.01  6140.3 1145.27
#Mann= 8 ,-1 , 0
  3289.3     .16       0  3418.3     .05       0  3739.6      .1       0
  4353.2     .05       0  4721.5     .16       0  4909.9      .1       0
  4948.7     .07       0  4954.7      .1       0
Bank Sta=4948.7,4954.7
XS Rating Curve= 0 ,0
Exp/Cntr=0.3,0.1

Type RM Length L Ch R = 1 ,7927    ,577,577,577
BEGIN DESCRIPTION:
Mapping XS c052af2c
END DESCRIPTION:
XS GIS Cut Line= 4
      2941731.68     10053446.22      2942975.62      10053515.6
      2943312.63      10053718.8      2944447.54     10053689.07
#Sta/Elev= 30
  3505.6 1132.42  3584.9 1127.87  3928.1 1116.25  4225.3 1108.82  4315.3 1105.41
  4403.8 1097.28  4548.9 1090.06    4564 1086.85  4604.1 1071.19  4634.1 1064.93
  4674.2 1061.69  4714.3 1065.62  4878.3 1057.64  4887.3  1057.2  4955.2 1051.16
  5004.6 1050.19  5007.3 1049.69  5010.6 1050.19  5137.1 1071.69  5173.5  1074.8
  5350.9 1080.48  5380.9 1083.66  5660.6 1091.24  5693.9 1092.97  5921.1 1110.05
  6001.1 1113.29  6061.2 1119.48  6121.2  1131.8  6251.2 1139.13  6280.3 1143.19
#Mann= 14 ,-1 , 0
  3505.6     .16       0  3584.9     .05       0  3928.1      .1       0
  4225.3     .16       0  4315.3      .1       0  4548.9     .05       0
  4878.3     .16       0  4887.3      .1       0  5004.6     .07       0
  5010.6      .1       0  5137.1     .05       0  5173.5      .1       0
  5660.6     .16       0  5693.9      .1       0
Bank Sta=5004.6,5010.6
XS Rating Curve= 0 ,0
Exp/Cntr=0.3,0.1

Type RM Length L Ch R = 1 ,7538    ,1715,1715,1715
BEGIN DESCRIPTION:
YEAGER CREEK 14.0
END DESCRIPTION:
XS GIS Cut Line= 4
      2941610.71     10053574.72      2942499.62     10053838.61
      2943756.57     10053748.34      2944525.46     10053672.14
#Sta/Elev= 30
  3638.8 1144.12  3714.9 1142.18  3811.5 1130.76  3933.9 1123.02  4110.9 1117.73
  4584.2 1101.69  4815.3 1094.12  4925.8 1087.27  4935.9 1083.36  4955.9 1066.85
 4979.55 1053.22  4987.1  1047.4    5003 1044.95  5005.8 1044.45    5009 1044.95
  5050.1 1046.47  5106.3 1052.34  5136.4 1056.79  5176.5 1062.05  5236.5 1063.73
  5240.1 1063.85  5344.2 1068.11  5429.9 1074.69  5647.7 1079.21    5888 1088.99
  5957.2 1093.71  6250.2 1113.49  6310.5 1119.49  6360.7  1131.8  6598.9 1150.09
#Mann= 16 ,-1 , 0
  3638.8      .1       0  3714.9     .16       0  3811.5     .05       0
  4110.9      .1       0  4584.2     .16       0  4815.3      .1       0
    5003     .07       0    5009      .1       0  5050.1     .05       0
  5136.4      .1       0  5236.5     .05       0  5240.1      .1       0
  5344.2     .05       0  5429.9      .1       0    5888     .16       0
  5957.2      .1       0
Bank Sta=4979.55,5106.3
XS Rating Curve= 0 ,0
Exp/Cntr=0.3,0.1

Type RM Length L Ch R = 1 ,7350    ,1527,1527,1527
BEGIN DESCRIPTION:
YEAGER CREEK 14.0
END DESCRIPTION:
XS GIS Cut Line= 4
      2941610.74     10053574.73      2942752.59     10053969.09
      2943352.28     10053951.74      2944523.97     10053743.66
#Sta/Elev= 30
  3505.5 1144.12    3583 1142.22    3679 1131.39  3788.5  1123.8  3974.9 1117.81
  4480.7 1100.54  4682.2 1093.73  4879.5 1087.95  4889.5 1084.53  4899.5 1069.49
  4919.5 1058.63  4959.5 1046.94  4986.5 1045.06  4989.3 1044.56  4992.5 1045.06
  5119.6 1062.61  5248.2 1065.29  5301.8 1065.44  5612.9 1064.73  5749.7 1080.15
  5790.1 1084.82  5899.3  1088.6  5934.6 1090.92  6021.4 1095.18  6129.3 1098.27
  6183.1 1105.53  6193.4 1109.56  6294.8 1116.54  6355.4 1133.27  6503.5 1146.74
#Mann= 14 ,-1 , 0
  3505.5      .1       0    3583     .16       0    3679     .05       0
  3974.9      .1       0  4480.7     .16       0  4682.2      .1       0
  4986.5     .07       0  4992.5      .1       0  5248.2     .05       0
  5301.8      .1       0  5749.7     .16       0  5899.3      .1       0
  5934.6     .16       0  6021.4      .1       0
Bank Sta=4986.5,4992.5
XS Rating Curve= 0 ,0
Exp/Cntr=0.3,0.1

Type RM Length L Ch R = 1 ,5823    ,1141,1141,1141
BEGIN DESCRIPTION:
YEAGER CREEK 11.0
END DESCRIPTION:
XS GIS Cut Line= 4
      2942541.33     10054088.63      2943610.73     10054512.23
      2944728.79      10054352.5      2944957.95     10054171.95
#Sta/Elev= 30
  3053.6 1098.67  3377.7 1093.57  3454.8 1090.76  3681.5 1086.49    3916 1079.75
  4160.2 1077.54  4282.2 1075.08    4356 1071.32  4625.8 1060.03  4809.8 1056.16
  4858.2 1054.27  4908.7 1045.55  4996.5 1037.15  5016.8  1036.9  5019.5  1036.4
  5022.8  1036.9    5040 1039.94  5050.1 1046.45  5070.3 1061.74  5076.2 1070.26
  5081.3 1068.65    5141 1112.59  5146.9 1118.74    5152 1117.92  5170.5 1129.32
  5217.6 1146.99    5482 1153.27  5517.3 1156.91  5543.2 1155.15    5625 1160.07
#Mann= 14 ,-1 , 0
  3053.6     .16       0  3377.7      .1       0  3454.8     .05       0
  3681.5      .1       0    3916     .05       0  4160.2      .1       0
  4282.2     .05       0    4356     .16       0  4809.8     .05       0
  4996.5     .16       0  5016.8     .07       0  5022.8     .16       0
  5170.5      .1       0  5543.2     .05       0
Bank Sta=4908.7,5050.1
XS Rating Curve= 0 ,0
Exp/Cntr=0.3,0.1

Type RM Length L Ch R = 1 ,4682    ,991,991,991
BEGIN DESCRIPTION:
YEAGER CREEK 9.0
END DESCRIPTION:
XS GIS Cut Line= 4
      2941742.67     10053810.83      2943284.34     10054588.61
      2943666.29     10055345.56       2943964.2     10055352.49
#Sta/Elev= 30
  2738.2 1134.81  2886.8 1123.44  3007.6 1119.37  3093.1 1115.98  3219.6 1110.95
  3257.8 1109.33  3330.8 1107.48  3452.7 1103.87  3871.8 1098.72  4045.6 1091.33
  4593.5 1083.11  4636.9 1082.64  4664.8 1078.78  4708.4 1065.56  4726.1 1059.26
  4761.9 1052.19  4830.8 1051.86  4908.1 1045.51  4932.4 1041.86  4946.5 1039.82
  4996.3 1036.37    4999 1035.87  5002.3 1036.37  5066.2 1041.89  5216.7 1065.19
  5266.9 1068.05  5309.7 1077.45  5442.9 1086.81    5495 1094.15  5610.8 1101.61
#Mann= 17 ,-1 , 0
  2738.2     .05       0  3007.6      .1       0  3093.1     .16       0
  3219.6      .1       0  3257.8     .16       0  3330.8      .1       0
  3452.7     .16       0  3871.8     .05       0  4045.6      .1       0
  4593.5     .16       0  4708.4      .1       0  4830.8     .16       0
  4908.1      .1       0  4946.5     .05       0  4996.3    .035       0
  5002.3     .05       0  5442.9      .1       0
Bank Sta=4932.4,5066.2
XS Rating Curve= 0 ,0
Exp/Cntr=0.3,0.1

Type RM Length L Ch R = 1 ,3691    ,811,811,811
BEGIN DESCRIPTION:
YEAGER CREEK 7.0
END DESCRIPTION:
XS GIS Cut Line= 4
      2941617.65     10053783.03      2942645.46     10054588.61
      2942569.07     10055144.17      2943033.93      10055511.9
#Sta/Elev= 30
    3373 1145.42  3480.8 1142.24  3509.7 1135.12  3588.3 1128.15  3794.7 1119.49
  4071.4 1106.63  4116.1 1106.27  4192.7  1104.6  4284.6    1102  4536.3 1093.85
  4684.1 1088.25  4696.3 1085.38  4744.1 1059.72  4774.9 1047.94  4885.9 1038.02
  5004.1 1029.16  5006.8 1028.66  5010.1 1029.16  5017.2    1030 5030.11  1038.4
  5040.3 1046.44  5056.5 1053.67  5151.2 1058.54    5264 1063.46  5424.1 1066.12
  5605.4 1074.07  5668.9  1077.2  5738.8 1081.14  5790.6 1082.64  5832.4 1084.55
#Mann= 17 ,-1 , 0
    3373     .05       0  3794.7      .1       0  4071.4     .16       0
  4116.1      .1       0  4192.7     .16       0  4284.6      .1       0
  4536.3     .16       0  4744.1     .05       0  5004.1    .035       0
  5010.1     .05       0  5040.3      .1       0  5151.2     .05       0
    5264      .1       0  5605.4     .05       0  5668.9      .1       0
  5738.8     .05       0  5790.6      .1       0
Bank Sta=4885.9,5030.11
XS Rating Curve= 0 ,0
Exp/Cntr=0.3,0.1

Type RM Length L Ch R = 1 ,2880    ,775,775,775
BEGIN DESCRIPTION:
YEAGER CREEK 5.0
END DESCRIPTION:
XS GIS Cut Line= 3
      2941284.34     10053921.94      2942006.57     10055109.45
      2942894.41     10055470.14
#Sta/Elev= 30
  3927.7 1160.08  3978.4 1158.99  4264.7 1144.94  4284.4 1144.54  4384.1 1141.56
  4411.3 1138.62  4442.3 1128.64  4524.7 1123.68  4606.4 1118.42  4696.1 1115.37
  4792.8 1105.43  4802.8 1104.21  4833.7 1095.13  4870.5 1089.03  4891.8 1072.48
  4907.3 1063.96  4944.1 1032.52  4973.7 1025.51  5014.7  1024.7  5017.4  1024.2
  5020.7  1024.7  5024.5  1024.9    5039 1025.01  5066.2 1033.09  5155.3 1041.31
  5373.9 1046.21  5446.1 1057.47  5535.5 1064.48  6029.8 1070.68  6275.9 1081.51
#Mann= 12 ,-1 , 0
  3927.7     .16       0  3978.4      .1       0  4264.7     .05       0
  4284.4      .1       0  4524.7     .05       0  4606.4      .1       0
  4792.8     .05       0  4802.8      .1       0  4973.7     .16       0
  5014.7     .07       0  5020.7     .16       0  5024.5      .1       0
Bank Sta=4944.1,5066.2
XS Rating Curve= 0 ,0
Exp/Cntr=0.3,0.1

Type RM Length L Ch R = 1 ,2105    ,635,635,635
BEGIN DESCRIPTION:
YEAGER CREEK 4.0
END DESCRIPTION:
XS GIS Cut Line= 4
      2941110.69     10055373.32      2941555.18     10055546.95
      2942430.18     10055331.67      2942812.14     10055526.12
#Sta/Elev= 30
  4168.1 1130.61  4337.5  1121.9  4459.4 1112.49    4520 1104.17  4584.2 1101.13
  4682.2 1098.13  4751.7 1094.03  4782.6  1090.5  4792.9 1087.28  4801.6 1080.81
  4806.8 1079.34  4843.2 1048.99  4848.3 1047.57  4854.6 1041.41  4875.2 1031.59
  4895.8 1026.97    4959 1023.84  5006.1 1019.63  5008.9 1019.13  5012.1 1019.63
  5029.7 1030.16  5055.9 1040.96  5144.1 1043.14  5180.5 1049.84    5222 1054.69
  5329.8 1062.92  5379.3 1064.62  5482.8 1068.12  5711.7 1069.97    5975 1081.02
#Mann= 7 ,-1 , 0
  4168.1      .1       0  4584.2     .05       0    4959      .1       0
  5006.1     .07       0  5012.1      .1       0  5329.8     .05       0
  5379.3      .1       0
Bank Sta=4875.2,5029.7
XS Rating Curve= 0 ,0
Exp/Cntr=0.3,0.1

Type RM Length L Ch R = 1 ,1470    ,725,725,725
BEGIN DESCRIPTION:
YEAGER CREEK 3.0
END DESCRIPTION:
XS GIS Cut Line= 4
       2941194.1     10055595.58      2941770.46     10055991.39
      2942506.57       10056165.      2942978.76     10056713.58
#Sta/Elev= 30
  3990.5  1120.8  4151.2 1110.07  4178.3 1102.94  4556.5 1092.85  4689.7 1087.19
  4770.1 1076.74  4821.2 1064.46  4831.5 1059.52  4849.6 1038.54  4854.8  1042.6
  4862.3 1033.95  4872.6 1029.48  4881.8  1027.6  5006.1 1019.83  5078.1 1029.97
  5088.3  1031.5  5108.7 1021.46  5116.2 1019.15  5118.9 1018.65  5122.2 1019.15
  5156.2 1030.21  5216.9  1031.9  5223.4  1031.9  5417.9 1033.22  5503.1 1046.55
  5549.7 1049.38  5638.5 1059.03  5879.4 1068.32    6021 1082.42  6169.8 1085.76
#Mann= 11 ,-1 , 0
  3990.5      .1       0  4556.5     .05       0  4881.8      .1       0
  5108.7     .16       0  5116.2     .07       0  5122.2     .16       0
  5216.9      .1       0  5223.4     .05       0  5417.9      .1       0
  5549.7     .05       0  5638.5      .1       0
#XS Ineff= 1 ,-1
 5087.12 5398.47 1031.25
Permanent Ineff=
       T
Bank Sta=4872.6,5078.1
XS Rating Curve= 0 ,0
Exp/Cntr=0.3,0.1

Type RM Length L Ch R = 1 ,745     ,513,513,513
BEGIN DESCRIPTION:
YEAGER CREEK 2.0
END DESCRIPTION:
XS GIS Cut Line= 4
      2941082.98     10055748.36      2941798.23     10056560.84
      2942221.84     10056963.61      2942971.83      10056977.5
#Sta/Elev= 30
  3670.6 1117.14  3820.2 1101.83  3971.9  1096.6  3989.4 1096.67  4110.5 1092.88
  4379.9  1064.9  4478.6  1061.3    4564 1046.61  4650.2  1039.7  4714.3 1037.44
  4826.2    1036  4903.9 1032.31  4939.2 1024.37  4953.3 1019.26  4999.7 1019.25
  5002.4 1018.75  5005.7 1019.25  5052.4  1020.4 5052.84 1025.83  5059.3 1029.71
  5115.9 1039.37  5186.7 1042.94  5286.8  1042.3  5434.2 1046.55  5504.2 1055.85
  5564.2 1055.09  5684.3 1060.94  5894.3 1083.86  6062.4 1092.25  6087.7 1092.85
#Mann= 10 ,-1 , 0
  3670.6      .1       0  3971.9     .16       0  3989.4      .1       0
  4650.2     .05       0  4714.3     .16       0  4826.2      .1       0
  4999.7     .07       0  5005.7      .1       0  5286.8     .16       0
  6062.4      .1       0
Bank Sta=4939.2,5052.84
XS Rating Curve= 0 ,0
Exp/Cntr=0.3,0.1

Type RM Length L Ch R = 1 ,232     ,0,0,0
BEGIN DESCRIPTION:
YEAGER CREEK 1.0
END DESCRIPTION:
XS GIS Cut Line= 4
      2940930.19     10055796.97      2941291.29      10056602.5
      2941617.68     10057019.17       2942742.7     10057505.29
#Sta/Elev= 30
  3775.9 1118.73  3855.9 1105.05  3982.1 1096.59  4052.3  1081.3  4108.6 1074.69
  4188.8 1066.21    4408 1056.79  4614.9 1040.88    4800 1031.88    4942 1017.13
  4957.7 1014.84  4996.8 1010.04  4999.5 1009.54  5002.8 1010.04  5120.1 1017.24
  5187.7 1029.78  5232.1 1032.95    5384 1032.52    5472 1024.05    5581  1029.6
  5635.3 1035.96  5669.7 1052.44    5679 1053.89  5711.3 1055.85  5821.6 1073.45
  5877.1 1075.31  5964.8 1079.95    6230 1086.76  6371.8 1089.59  6413.5 1090.85
#Mann= 11 ,-1 , 0
  3775.9      .1       0  3982.1     .16       0  4108.6      .1       0
  4614.9     .16       0  4957.7      .1       0  4996.8     .07       0
  5002.8      .1       0  5877.1     .16       0  5964.8      .1       0
    6230     .05       0  6371.8      .1       0
#XS Ineff= 2 , 0
                         5240.34         1033.19
Permanent Ineff=
       T       T
Bank Sta=4942,5120.1
XS Rating Curve= 0 ,0
Exp/Cntr=0.3,0.1

Chan Stop Cuts=-1
Use User Specified Reach Order=0
Composite Channel Slope=5
